--- Black Creek.prj (project) ---

Proj Title=Black Creek Base Level Engineering
Current Plan=p02
Default Exp/Contr=0.3,0.1
English Units
Geom File=g01
Flow File=f01
Plan File=p02
Y Axis Title=Elevation
X Axis Title(PF)=Main Channel Distance
X Axis Title(XS)=Station
BEGIN DESCRIPTION:
Black Creek
END DESCRIPTION:
DSS File=dss
DSS Export Rating Curves= 0
DSS Export Rating Curve Sorted= 0
DSS Export Volume Flow Curves= 0
DXF OffsetX= 0
DXF OffsetY= 0
DXF ScaleX= 1
DXF ScaleY= 10

--- Black Creek.p02 (plan) ---

Plan Title=Multiple Plan
Program Version=5.07
Short Identifier=Multiple Plan
Geom File=g01
Flow File=f01
Subcritical Flow
K Sum by GR= 0
Std Step Tol= 0.01
Critical Tol= 0.01
Num of Std Step Trials= 20
Max Error Tol= 0.3
Flow Tol Ratio= 0.001
Split Flow NTrial= 30
Split Flow Tol= 0.02
Split Flow Ratio= 0.02
Log Output Level= 0
Friction Slope Method= 1
Unsteady Friction Slope Method= 2
Unsteady Bridges Friction Slope Method= 1
Parabolic Critical Depth
Global Vel Dist= 1 , 1 , 1
Global Log Level= 0
CheckData=True
Encroach Param=-1 ,0,0, 0
BEGIN DESCRIPTION:
Multiple Run
END DESCRIPTION:
Computation Interval=1MIN
Output Interval=1HOUR
Instantaneous Interval=1HOUR
Mapping Interval=1HOUR
Computation Time Step Use Courant=        0
Computation Time Step Use Time Series=    0
Computation Time Step Count To Double=0
Computation Time Step Max Doubling=0
Computation Time Step Max Halving=0
Computation Time Step Residence Courant=0
Run HTab= 0
Run UNet= 0
Run Sediment= 0
Run PostProcess= 0
Run WQNet= 0
Run RASMapper= 0
UNET Theta= 1
UNET Theta Warmup= 1
UNET ZTol= 0.02
UNET ZSATol= 0.02
UNET MxIter= 20
UNET Max Iter WO Improvement= 0
UNET MaxInSteps= 0
UNET DtIC= 0
UNET DtMin= 0
UNET MaxCRTS= 20
UNET WFStab= 2
UNET SFStab= 1
UNET WFX= 1
UNET SFX= 1
UNET 1D Methodology=Finite Difference
UNET DSS MLevel= 4
UNET Pardiso=0
UNET DZMax Abort= 100
UNET Use Existing IB Tables=-1
UNET Froude Reduction=False
UNET Froude Limit= 0.8
UNET Froude Power= 4
UNET D1 Cores= 0
UNET D2 Coriolis=0
UNET D2 Cores= 0
UNET D2 Theta= 1
UNET D2 Theta Warmup= 1
UNET D2 Z Tol= 0.01
UNET D2 Volume Tol= 0.01
UNET D2 Max Iterations= 20
UNET D2 Equation= 0
UNET D2 RampUpFraction=0.1
UNET D2 TimeSlices= 1
UNET D2 BCVolumeCheck=0
UNET D1D2 MaxIter= 0
UNET D1D2 ZTol=0.01
UNET D1D2 QTol=0.1
UNET D1D2 MinQTol=1
DSS File=dss
Write IC File= 0
Write IC File at Fixed DateTime=0
Write IC File at Sim End=0
Echo Input=False
Echo Parameters=False
Echo Output=False
Write Detailed= 0
HDF Write Warmup=0
HDF Write Time Slices=0
HDF Flush=0
HDF Face Node Velocities=0
HDF Compression= 1
HDF Chunk Size= 1
HDF Spatial Parts= 1
HDF Use Max Rows=0
HDF Fixed Rows= 1
Calibration Method= 0
Calibration Iterations= 20
Calibration Max Change=0.05
Calibration Tolerance=0.2
Calibration Maximum=1.5
Calibration Minimum=0.5
Calibration Optimization Method= 1
WQ AD Non Conservative
WQ ULTIMATE=-1
WQ Max Comp Step=1HOUR
WQ Output Interval=15MIN
WQ Output Selected Increments= 0
WQ Output face flow=0
WQ Output face velocity=0
WQ Output face area=0
WQ Output face dispersion=0
WQ Output cell volume=0
WQ Output cell surface area=0
WQ Output cell continuity=0
WQ Output cumulative cell continuity=0
WQ Output face conc=0
WQ Output face dconc_dx=0
WQ Output face courant=0
WQ Output face peclet=0
WQ Output face adv mass=0
WQ Output face disp mass=0
WQ Output cell mass=0
WQ Output cell source sink temp=0
WQ Output nsm pathways=0
WQ Output nsm derived pathways=0
WQ Output MaxMinRange=-1
WQ Daily Max Min Mean=-1
WQ Daily Range=0
WQ Daily Time=0
WQ Create Restart=0
WQ Fixed Restart=0
WQ System Summary=0
WQ Write To DSS=0
WQ Use Fixed Temperature=0
Sorting and Armoring Iterations= 10
XS Update Threshold= 0.02
Bed Roughness Predictor= 0
Hydraulics Update Threshold= 0.02
Energy Slope Method= 1
Volume Change Method= 1
Sediment Retention Method= 0
XS Weighting Method= 0
Number of US Weighted Cross Sections= 1
Number of DS Weighted Cross Sections= 1
Upstream XS Weight=0
Main XS Weight=1
Downstream XS Weight=0
Number of DS XS's Weighted with US Boundary= 1
Upstream Boundary Weight= 1
Weight of XSs Associated with US Boundary= 0
Number of US XS's Weighted with DS Boundary= 1
Downstream Boundary Weight= 0.5
Weight of XSs Associated with DS Boundary= 0.5
Percentile Method= 0
Sediment Output Level= 3
Mass or Volume Output= 0
Output Increment Type= 1
Profile and TS Output Increment= 1
XS Output Flag= 0
XS Output Increment= 10
Write Gradation File= 0
Read Gradation Hotstart= 0
Write HDF5 File= 1
Write Binary Output= 1
Write DSS Sediment File= 0
SV Curve= 0
Specific Gage Flag= 0

--- Black Creek.f01 (steady flow) ---

Flow Title=Multiple
Program Version=5.05
Number of Profiles= 7
Profile Names=10-year,25-year,50-year,1pct_min,100-year,1pct_plu,500-year
River Rch & RM=Black Creek,Reach-1         ,220601
     491     675     825     499     996    1988    1457
River Rch & RM=Black Creek,Reach-1         ,218938
     751    1059    1315     808    1612    3216    2430
River Rch & RM=Black Creek,Reach-1         ,215309
     989    1413    1771    1096    2187    4364    3350
River Rch & RM=Black Creek,Reach-1         ,209097
    1087    1561    1963    1219    2432    4852    3748
River Rch & RM=Black Creek,Reach-1         ,206605
    1219    1760    2221    1384    2761    5509    4284
River Rch & RM=Black Creek,Reach-1         ,203188
    1929    2840    3632    2288    4566    9110    7248
River Rch & RM=Black Creek,Reach-1         ,196560
    2047    3020    3867    2440    4868    9713    7746
River Rch & RM=Black Creek,Reach-1         ,195989
    2354    3491    4486    2839    5664   11300    9067
River Rch & RM=Black Creek,Reach-1         ,185872
    2394    3546    4553    2879    5744   11460    9180
River Rch & RM=Black Creek,Reach-1         ,182454
    2590    3852    4961    3145    6275   12520   10083
River Rch & RM=Black Creek,Reach-1         ,180161
    2659    3953    5088    3223    6430   12829   10316
River Rch & RM=Black Creek,Reach-1         ,175419
    2861    4267    5504    3493    6970   13907   11229
River Rch & RM=Black Creek,Reach-1         ,171121
    4367    6601    8593    5498   10969   21886   17948
River Rch & RM=Black Creek,Reach-1         ,169073
    4367    6601    8593    5498   10969   21886   17948
River Rch & RM=Black Creek,Reach-1         ,161260
    4367    6601    8593    5498   10969   21886   17948
River Rch & RM=Black Creek,Reach-1         ,159686
    4367    6601    8593    5498   10969   21886   17948
River Rch & RM=Black Creek,Reach-1         ,151262
    4367    6601    8593    5498   10969   21886   17948
River Rch & RM=Black Creek,Reach-1         ,145664
    4467    6750    8786    5619   11212   22370   18334
River Rch & RM=Black Creek,Reach-1         ,142105
    4564    6898    8981    5745   11464   22873   18754
River Rch & RM=Black Creek,Reach-1         ,139488
    4739    7171    9342    5979   11930   23804   19538
River Rch & RM=Black Creek,Reach-1         ,134083
    5409    8217   10733    6885   13738   27410   22593
River Rch & RM=Black Creek,Reach-1         ,132832
    5409    8217   10733    6885   13738   27410   22593
River Rch & RM=Black Creek,Reach-1         ,129709
    5515    8377   10941    7018   14002   27939   23024
River Rch & RM=Black Creek,Reach-1         ,128535
    5515    8377   10941    7018   14002   27939   23024
River Rch & RM=Black Creek,Reach-1         ,123956
    5550    8425   11000    7052   14070   28074   23112
River Rch & RM=Black Creek,Reach-1         ,117346
    5605    8505   11100    7113   14193   28319   23298
River Rch & RM=Black Creek,Reach-1         ,110146
    5953    9050   11826    7587   15138   30204   24902
River Rch & RM=Black Creek,Reach-1         ,108978
    5953    9050   11826    7587   15138   30204   24902
River Rch & RM=Black Creek,Reach-1         ,107706
    6025    9159   11969    7679   15322   30571   25206
River Rch & RM=Black Creek,Reach-1         ,103858
    6064    9216   12042    7724   15412   30750   25344
River Rch & RM=Black Creek,Reach-1         ,100659
    6134    9325   12187    7818   15600   31126   25661
River Rch & RM=Black Creek,Reach-1         ,95677
    6130    9316   12173    7808   15579   31084   25617
River Rch & RM=Black Creek,Reach-1         ,94139
    6986   10650   13943    8958   17873   35661   29474
River Rch & RM=Black Creek,Reach-1         ,90453
    7642   11675   15309    9848   19649   39206   32490
River Rch & RM=Black Creek,Reach-1         ,80482
    7642   11675   15309    9848   19649   39206   32490
River Rch & RM=Black Creek,Reach-1         ,74433
    7642   11675   15309    9848   19649   39206   32490
River Rch & RM=Black Creek,Reach-1         ,70286
    7560   11545   15134    9735   19425   38758   32122
River Rch & RM=Black Creek,Reach-1         ,68046
    7285   11099   14536    9353   18662   37235   30929
River Rch & RM=Black Creek,Reach-1         ,65587
    7285   11099   14536    9353   18662   37235   30929
River Rch & RM=Black Creek,Reach-1         ,56661
    7285   11099   14536    9353   18662   37235   30929
River Rch & RM=Black Creek,Reach-1         ,45499
    7285   11099   14536    9353   18662   37235   30929
River Rch & RM=Black Creek,Reach-1         ,42779
    6845   10400   13600    8747   17453   34823   28941
River Rch & RM=Black Creek,Reach-1         ,38978
    6831   10377   13568    8726   17410   34737   28865
River Rch & RM=Black Creek,Reach-1         ,35100
    6765   10265   13412    8620   17199   34318   28483
River Rch & RM=Black Creek,Reach-1         ,30185
    6732   10209   13334    8568   17094   34108   28294
River Rch & RM=Black Creek,Reach-1         ,28439
    6732   10209   13334    8568   17094   34108   28294
River Rch & RM=Black Creek,Reach-1         ,18600
    6382    9653   12593    8096   16154   32232   26827
River Rch & RM=Black Creek,Reach-1         ,11987
    6382    9650   12588    8092   16145   32214   26809
River Rch & RM=Black Creek,Reach-1         ,9113
    6382    9650   12588    8092   16145   32214   26809
Boundary for River Rch & Prof#=Black Creek,Reach-1         , 1
Up Type= 0
Dn Type= 3
Dn Slope=0.00063
Boundary for River Rch & Prof#=Black Creek,Reach-1         , 2
Up Type= 0
Dn Type= 3
Dn Slope=0.00063
Boundary for River Rch & Prof#=Black Creek,Reach-1         , 3
Up Type= 0
Dn Type= 3
Dn Slope=0.00063
Boundary for River Rch & Prof#=Black Creek,Reach-1         , 4
Up Type= 0
Dn Type= 3
Dn Slope=0.00063
Boundary for River Rch & Prof#=Black Creek,Reach-1         , 5
Up Type= 0
Dn Type= 3
Dn Slope=0.00063
Boundary for River Rch & Prof#=Black Creek,Reach-1         , 6
Up Type= 0
Dn Type= 3
Dn Slope=0.00063
Boundary for River Rch & Prof#=Black Creek,Reach-1         , 7
Up Type= 0
Dn Type= 3
Dn Slope=0.00063
DSS Import GetInterval= 0
DSS Import GetPeak= 0
DSS Import FillOption= 0

--- Black Creek.g01 (geometry) ---

Geom Title=Black Creek
Program Version=5.07

River Reach=Black Creek     ,Reach-1
Reach XY= 30
      1973207.44     13648188.72      1972716.72     13640794.44
       1973850.8     13639144.54       1971240.8     13634744.54
       1973160.8     13631134.54       1972270.8     13620474.54
       1973960.8     13618104.54       1972130.8     13610584.54
      1973641.56     13605892.76       1975400.8     13604814.54
       1975130.8     13596894.54       1973330.8     13595384.54
       1974960.8     13591424.54       1973240.8     13588904.54
       1972680.8     13582504.54       1974930.8     13580864.54
       1976700.8     13581354.54        1976451.     13575932.44
       1977910.8     13574074.54       1974400.8     13565754.54
       1973610.8     13556014.54       1975520.8     13552724.54
       1972380.8     13548114.54       1972370.8     13543674.54
       1977030.8     13536094.54       1978000.8     13528464.54
      1981462.13     13525979.05       1984230.8     13520464.54
       1985600.8     13510784.54      1995135.29     13499801.48

Type RM Length L Ch R = 1 ,220601  ,460,460,460
BEGIN DESCRIPTION:
Mapping XS 6efbf12d
END DESCRIPTION:
XS GIS Cut Line= 3
      1973748.28     13647969.54       1973289.9     13647966.07
       1972598.6     13648180.91
#Sta/Elev= 30
  4374.9  919.75  4528.2  916.88  4558.2  915.71  4578.2  915.71  4598.2  914.54
  4678.2  912.79  4688.2   912.1  4708.2  911.96  4818.2  908.54  4850.3  907.88
  4872.7  907.99    4948  906.84    4957   904.5  4964.1  903.16  4980.6  898.92
  4992.5  898.74    4993  897.94    4998  897.94  4998.5  898.74    5006  898.81
  5018.3  900.96  5121.2  902.47    5163  902.66  5257.3  904.59  5278.2  904.15
  5333.2  906.14  5424.5  909.17  5477.2  911.11  5517.1  913.39  5557.2  913.49
#Mann= 7 ,-1 , 0
  4374.9      .1       0  4872.7     .16       0    4957      .1       0
  4992.5     .07       0  4998.5      .1       0  5333.2     .05       0
  5424.5      .1       0
Bank Sta=4992.5,4998.5
XS Rating Curve= 0 ,0
Exp/Cntr=0.3,0.1

Type RM Length L Ch R = 1 ,220141  ,253,253,253
BEGIN DESCRIPTION:
Black Creek 240.0
END DESCRIPTION:
XS GIS Cut Line= 3
      1973710.92     13647695.67      1973110.22     13647647.06
      1972492.13      13647692.2
#Sta/Elev= 30
  4244.2  915.07  4260.2  914.88  4270.2  913.88  4314.9  912.24  4350.5   911.2
  4370.5  911.27  4442.1  908.42  4571.2  905.21  4661.5  904.13  4686.5  903.28
  4751.8  902.89  4808.7  901.03  4868.7  900.29  4904.5   900.1  4979.4  899.41
  4979.9  898.61  4984.9  898.61  4985.4  899.41  5002.5  899.94  5021.1   901.7
  5026.1  901.57  5032.6  902.54  5052.6  903.44  5102.8  903.41    5203  901.16
  5263.2   901.9  5313.3  903.83  5343.4  906.97  5393.5  907.85  5466.6  911.07
#Mann= 5 ,-1 , 0
  4244.2      .1       0  4868.7     .16       0  4904.5      .1       0
  4979.4     .07       0  4985.4      .1       0
Bank Sta=4979.4,4985.4
XS Rating Curve= 0 ,0
Exp/Cntr=0.3,0.1

Type RM Length L Ch R = 1 ,219888  ,42,42,42
BEGIN DESCRIPTION:
Mapping XS c5d4dc9e
END DESCRIPTION:
XS GIS Cut Line= 4
       1973738.3     13647423.97      1973293.38     13647413.12
      1972713.95      13647465.2      1972464.38     13647467.37
#Sta/Elev= 30
  4140.7  910.62    4184   909.8    4194  908.95    4214  908.67  4301.2  905.64
  4314.1  905.42  4324.1  905.93  4344.1  904.73  4374.1  903.98  4424.1   902.9
  4454.1  902.79  4534.1  901.34  4574.1  900.24  4585.8  900.38  4604.2  899.37
  4614.2  899.99  4644.4  899.38  4754.8  898.53  4777.1  898.87  4845.2  898.23
  4888.2  898.63  4925.5  898.26  4982.7  896.02  4983.2  895.22  4988.2  895.22
  4988.7  896.02  5076.1  897.31  5256.5   904.6  5296.5  906.74  5417.1  909.32
#Mann= 3 ,-1 , 0
  4140.7     .05       0  4982.7     .04       0  4988.7     .05       0
Bank Sta=4982.7,4988.7
XS Rating Curve= 0 ,0
Exp/Cntr=0.3,0.1

Type RM Length L Ch R = 1 ,219846  ,418,418,418
BEGIN DESCRIPTION:
Mapping XS 128b270e
END DESCRIPTION:
XS GIS Cut Line= 4
      1973731.77     13647397.93      1973289.04     13647378.39
      1972713.95     13647428.31       1972468.3       13647424.
#Sta/Elev= 30
  4157.1  910.23  4223.9  907.99    4264  907.15    4294  905.86    4333   905.1
  4344.1  904.46  4464.2   902.4  4494.2  901.44  4544.2  901.07  4594.3  900.05
  4599.8  898.87  4619.1  899.75    4795  898.02  4915.5  898.22  4963.2  896.99
  4968.2  897.36  4975.7  897.04  4982.7  895.33  4983.2  894.53  4988.2  894.53
  4988.7  895.33  5035.9  895.84    5066  896.64  5186.5   901.2  5216.5  902.85
  5236.5  903.21  5266.5  904.52  5286.5  906.19  5356.5   906.9  5423.2  909.91
#Mann= 3 ,-1 , 0
  4157.1     .05       0  4982.7     .04       0  4988.7     .05       0
Bank Sta=4982.7,4988.7
XS Rating Curve= 0 ,0
Exp/Cntr=0.3,0.1

Type RM Length L Ch R = 1 ,219428  ,490,490,490
BEGIN DESCRIPTION:
Black Creek 239.0
END DESCRIPTION:
XS GIS Cut Line= 3
      1973713.52     13647082.39      1973317.25     13647042.02
      1972555.52     13646990.37
#Sta/Elev= 30
  4154.2     910  4233.1  908.14  4263.3  907.01  4272.4  906.07  4277.4  906.35
  4313.5  904.95  4357.2  902.19    4372  901.12  4444.2  898.53  4524.6  896.95
  4544.7  897.57  4586.1  896.25  4624.9  896.24  4695.1  895.06  4715.1  895.31
  4955.7  894.44  4975.7  893.87  4992.8  892.23  4993.3  891.43  4998.3  891.43
  4998.8  892.23  5015.8  894.02  5126.1  896.58  5196.2  898.84  5226.3  901.68
  5236.7  902.09  5266.4  903.72  5276.4  904.79  5286.5  903.91    5316   905.8
#Mann= 5 ,-1 , 0
  4154.2     .16       0  4357.2      .1       0  4992.8     .07       0
  4998.8      .1       0  5236.7     .05       0
Bank Sta=4992.8,4998.8
XS Rating Curve= 0 ,0
Exp/Cntr=0.3,0.1

Type RM Length L Ch R = 1 ,218938  ,51,51,51
BEGIN DESCRIPTION:
Mapping XS e0f0b007
END DESCRIPTION:
XS GIS Cut Line= 4
      1973832.46     13646728.23      1973491.27     13646723.02
      1973043.36     13646712.61      1972441.76     13646699.58
#Sta/Elev= 30
  4298.1  910.68  4400.4  907.71  4495.6  905.44  4565.6  901.79  4605.6  900.97
  4725.6  897.07    4765  895.03    4770  895.48  4775.6  894.67  4795.6  893.91
  4845.7  892.96  4905.7   893.1  4982.7  892.31  4983.2  891.51  4988.2  891.51
  4988.7  892.31  5055.7  893.32  5204.3  893.03  5209.3  894.83  5265.8  895.36
  5305.8  896.52  5375.8  900.29  5435.8  900.64  5485.2   901.7  5535.8  903.57
  5555.8  905.03  5565.8  904.54  5579.2  905.12  5649.3  907.85  5689.1  909.07
#Mann= 7 ,-1 , 0
  4298.1     .16       0  4400.4      .1       0  4982.7     .07       0
  4988.7      .1       0  5485.2     .05       0  5579.2      .1       0
  5649.3     .05       0
Bank Sta=4982.7,4988.7
XS Rating Curve= 0 ,0
Exp/Cntr=0.3,0.1

Type RM Length L Ch R = 1 ,218887  ,40,40,40
BEGIN DESCRIPTION:
Mapping XS e8bd99a7
END DESCRIPTION:
XS GIS Cut Line= 3
       1973811.6     13646699.59      1972907.94     13646665.73
      1972433.94     13646663.13
#Sta/Elev= 30
  4348.1  909.81  4403.8     908  4437.1  906.89  4514.8  904.02  4524.8   904.5
  4634.9  899.42  4704.9  898.51    4785  895.83    4795  895.39    4802  891.06
  4802.5  890.26  4807.5  890.26    4808  891.06    4815  891.96    4825  894.39
  4855.1  893.06  4995.2  892.49  5005.2  893.08  5045.2  898.53  5065.2  900.55
  5085.2  901.77  5139.3  903.37  5425.3  905.14  5525.3  903.57  5552.2  903.76
  5585.3  905.17  5596.7  905.04  5605.3  904.77  5705.7  908.43  5726.4  909.22
#Mann= 8 ,-1 , 0
  4348.1      .1       0  4403.8     .16       0  4437.1      .1       0
    4802     .07       0    4808      .1       0  5552.2     .05       0
  5596.7      .1       0  5705.7     .05       0
Bank Sta=4802,4808
XS Rating Curve= 0 ,0
Exp/Cntr=0.3,0.1

Type RM Length L Ch R = 1 ,218847  ,282,282,282
BEGIN DESCRIPTION:
Black Creek 238.0
END DESCRIPTION:
XS GIS Cut Line= 3
       1973819.4     13646637.08      1973355.22     13646635.65
       1972445.5     13646634.78
#Sta/Elev= 30
  4341.4  909.53  4415.8  907.56  4439.1  906.54  4465.8  905.02  4557.1  901.32
  4575.8  901.04  4615.8  899.07  4695.8  895.92  4725.8  895.31  4755.8  895.38
  4803.2  893.34  4865.8  892.77  4905.8  891.77  4972.7  891.33  4973.2  890.53
  4978.3  890.53  4978.8  891.33  4995.8  891.43  5005.8  891.85  5055.8  892.01
  5155.8  891.66  5255.8  891.91  5425.8  898.64  5515.8  901.77  5555.8  902.77
    5580  903.92  5588.1  904.56  5595.8  905.23  5605.8  904.94  5715.3  908.49
#Mann= 7 ,-1 , 0
  4341.4      .1       0  4439.1     .16       0  4557.1      .1       0
  4972.7     .07       0  4978.8      .1       0    5580     .05       0
  5588.1      .1       0
Bank Sta=4972.7,4978.8
XS Rating Curve= 0 ,0
Exp/Cntr=0.3,0.1

Type RM Length L Ch R = 1 ,218565  ,310,310,310
BEGIN DESCRIPTION:
Mapping XS 661f908f
END DESCRIPTION:
XS GIS Cut Line= 3
      1973681.37     13646475.63      1973301.17      13646457.4
      1972764.68     13646173.53
#Sta/Elev= 30
  4476.4  910.33  4542.8   907.1  4627.7  899.99    4643   898.1    4703  893.15
  4800.4  891.14  4823.2  891.47  4833.2  890.52  4975.6  889.12  4981.3  888.79
  4985.4  886.61  4985.9  885.81    4991  885.81  4991.5  886.61  5003.3  888.74
  5101.6  890.93    5146  892.78    5190  893.35    5278  897.74  5293.9  898.97
    5322  903.33  5327.9  905.23  5338.4  907.01    5344  907.09  5360.4  910.07
    5366  910.19  5382.4  913.43  5388.1  913.22  5432.1  917.34    5464  918.82
#Mann= 4 ,-1 , 0
  4476.4     .16       0  4627.7      .1       0  4985.4     .07       0
  4991.5      .1       0
Bank Sta=4985.4,4991.5
XS Rating Curve= 0 ,0
Exp/Cntr=0.3,0.1

Type RM Length L Ch R = 1 ,218255  ,519,519,519
BEGIN DESCRIPTION:
Black Creek 237.0
END DESCRIPTION:
XS GIS Cut Line= 3
      1973725.01       13646325.        1973325.       13646225.
      1972975.01       13646075.
#Sta/Elev= 30
  4649.8  912.34  4701.4  910.76  4750.3  905.92  4755.5  906.21  4763.2  904.96
  4796.7  902.75  4832.8  898.13  4844.4  897.38    4874  893.09  4897.2  891.39
  4969.4  889.17  4994.7  885.16  4995.2  884.36  5000.3  884.36  5000.8  885.16
  5002.9  886.54  5010.6  887.03  5031.2  886.85  5038.9  885.86  5044.1  888.19
  5051.8  888.52  5071.2  888.99  5105.6  888.21  5205.4  889.73  5281.5  892.43
  5312.4  894.52    5345  897.92  5381.3  903.05  5410.3  908.26  5442.9  910.84
#Mann= 4 ,-1 , 0
  4649.8     .16       0  4844.4      .1       0  4994.7     .07       0
  5000.8      .1       0
Bank Sta=4994.7,5000.8
XS Rating Curve= 0 ,0
Exp/Cntr=0.3,0.1

Type RM Length L Ch R = 1 ,217736  ,52,52,52
BEGIN DESCRIPTION:
Black Creek 236.0
END DESCRIPTION:
XS GIS Cut Line= 4
      1974081.57     13645672.66       1973472.2     13645743.84
      1973395.81     13645974.75      1972994.41     13645869.85
#Sta/Elev= 30
  4313.6  903.19  4370.6  900.89  4410.8  898.06  4547.1  891.41  4631.3  887.26
  4692.7  887.33  4702.8  889.83    4733  892.35  4891.5  889.16  4930.4  889.07
  4949.4  888.19  4959.9  887.06  4965.6  885.56    4981  884.68  4988.4  882.06
  4988.9  881.26  4994.1  881.26  4994.6  882.06  4997.3  882.33  5002.6   884.6
  5054.7  886.34  5187.9  887.01  5263.6  886.36  5367.5  890.09  5390.1  891.76
  5425.4  896.54  5460.6  898.03  5481.2  902.23  5512.2  906.92  5585.2   913.2
#Mann= 4 ,-1 , 0
  4313.6      .1       0  4547.1     .16       0  4988.4     .07       0
  4994.6      .1       0
Bank Sta=4988.4,4994.6
XS Rating Curve= 0 ,0
Exp/Cntr=0.3,0.1

Type RM Length L Ch R = 1 ,217684  ,198,198,198
BEGIN DESCRIPTION:
Mapping XS e00b7afa
END DESCRIPTION:
XS GIS Cut Line= 4
      1974074.76     13645650.09      1973435.39     13645698.27
      1973367.68     13645930.04      1973009.19     13645837.82
#Sta/Elev= 30
  4277.5  903.45  4347.5  900.75  4417.7  895.99  4502.2  891.68  4537.7  890.76
  4598.2  887.01  4648.3  887.34  4668.4  889.51  4674.5  891.01  4679.5  889.74
  4698.4  891.49  4897.9  888.28  4934.4  888.38  4978.3  882.96  4995.5  882.24
    4996  881.44  5001.2  881.44  5001.7  882.24  5011.7  884.86  5193.9  886.25
  5321.9  889.46  5357.5  893.58  5410.7   896.9    5421   898.2  5438.9  903.25
  5444.1  902.47    5452  904.58  5479.6  908.64  5484.8  908.34  5530.3  912.47
#Mann= 5 ,-1 , 0
  4277.5      .1       0  4502.2     .16       0  4897.9      .1       0
  4995.5     .07       0  5001.7      .1       0
Bank Sta=4995.5,5001.7
XS Rating Curve= 0 ,0
Exp/Cntr=0.3,0.1

Type RM Length L Ch R = 1 ,217486  ,777,777,777
BEGIN DESCRIPTION:
Black Creek 235.0
END DESCRIPTION:
XS GIS Cut Line= 3
      1973983.09     13645501.66      1973475.32      13645592.8
      1972982.66     13645675.27
#Sta/Elev= 30
  4348.4  902.01  4447.6     893  4506.4   890.5  4589.2  889.03  4630.9  887.51
  4651.3  885.54  4661.4  883.65  4671.6  883.27  4682.7     885  4731.3  884.71
    4763  887.93  4803.7  887.93  4861.9  885.21  4909.1  885.83  4969.8  885.17
  4993.3  881.74  4993.8  880.94    4999  880.94  4999.5  881.74  5006.6  883.44
  5016.7  884.05  5047.9  884.58  5212.6  892.02  5229.6  894.03    5260  895.82
  5268.2  897.36  5273.3  896.79    5334  905.18  5341.2  906.92  5363.8  909.16
#Mann= 5 ,-1 , 0
  4348.4      .1       0  4589.2     .16       0  4993.3     .07       0
  4999.5     .16       0  5047.9      .1       0
Bank Sta=4993.3,4999.5
XS Rating Curve= 0 ,0
Exp/Cntr=0.3,0.1

Type RM Length L Ch R = 1 ,216709  ,335,335,335
BEGIN DESCRIPTION:
Black Creek 234.0
END DESCRIPTION:
XS GIS Cut Line= 3
      1974059.11     13645186.99        1973525.       13645125.
      1972885.01     13645087.16
#Sta/Elev= 30
  4458.1  899.19  4492.4  896.96  4606.8  892.42  4623.3  890.97  4643.4  890.83
  4663.6  889.28  4713.9  887.65    4734  885.84  4744.1  886.75  4828.5  884.96
    4875  884.25  4895.1  883.08  4945.5  882.87  4985.7  879.87  4993.3  877.29
  5002.6  876.96  5003.1  876.16  5008.6  876.16  5009.1  876.96  5015.8  877.27
  5055.9  882.43  5085.9  884.13  5098.2  884.13    5145  883.81  5266.3  884.02
  5296.3  884.76  5316.4  884.22  5391.3  885.94  5486.6  888.35  5636.9  895.14
#Mann= 7 ,-1 , 0
  4458.1      .1       0  4828.5     .16       0  5002.6     .07       0
  5009.1     .16       0  5098.2      .1       0    5145     .16       0
  5391.3      .1       0
Bank Sta=5002.6,5009.1
XS Rating Curve= 0 ,0
Exp/Cntr=0.3,0.1

Type RM Length L Ch R = 1 ,216374  ,259,259,259
BEGIN DESCRIPTION:
Black Creek 233.0
END DESCRIPTION:
XS GIS Cut Line= 3
       1974460.4     13645258.26      1973684.37     13644838.99
      1972694.83      13644784.3
#Sta/Elev= 30
  4064.3  916.84  4218.2  911.26  4286.4  910.93    4352  908.87  4388.7  906.52
  4417.7  902.89  4439.6  903.04  4477.7  900.78  4543.3  898.79  4587.1  898.64
  4625.2  895.91  4647.1  893.08  4706.9  888.78    4741  884.85  4809.2  880.84
  4898.3  880.53  4934.3  885.63  4982.5  875.99    4983  875.19  4988.5  875.19
    4989  875.99  5055.9  881.95  5075.9  882.14    5126  880.41  5314.5  882.94
  5466.5  885.69  5652.3  892.11  5676.8   893.1  5716.9  892.91  5937.4  902.16
#Mann= 5 ,-1 , 0
  4064.3      .1       0  4982.5     .07       0    4989      .1       0
  5314.5     .05       0  5652.3      .1       0
Bank Sta=4982.5,4989
XS Rating Curve= 0 ,0
Exp/Cntr=0.3,0.1

Type RM Length L Ch R = 1 ,216115  ,721,721,721
BEGIN DESCRIPTION:
Black Creek 232.0
END DESCRIPTION:
XS GIS Cut Line= 5
      1974603.66     13644615.03       1973895.3     13644664.51
      1973673.95     13644604.61      1973465.62     13644635.86
      1972634.92     13644677.53
#Sta/Elev= 30
  4082.9  918.24  4221.9   914.8  4312.1  911.19  4392.3  904.83  4472.5   900.8
  4492.6  898.77  4532.7  900.57  4552.7  897.96  4581.3  896.47  4612.8  899.12
  4652.9  894.01  4723.1  890.05  4809.5  879.89  4884.1  878.83  4907.3  875.75
  4923.9  875.15  4925.8  874.08  4926.3  873.28  4931.9  873.28  4932.4  874.08
  4958.6  875.08  4963.8  874.14  4998.5  874.61  5019.2  878.32  5074.2  880.01
  5243.6  880.65  5363.7  883.63    5564  886.42  5877.2  895.15  6064.7  903.18
#Mann= 5 ,-1 , 0
  4082.9      .1       0  4925.8     .07       0  4932.4      .1       0
  5074.2     .05       0  5877.2      .1       0
Bank Sta=4925.8,4932.4
XS Rating Curve= 0 ,0
Exp/Cntr=0.3,0.1

Type RM Length L Ch R = 1 ,215394  ,85,85,85
BEGIN DESCRIPTION:
Mapping XS 2b180b80
END DESCRIPTION:
XS GIS Cut Line= 6
        1974575.     13643656.69      1973791.14     13643865.03
      1973634.89      13643846.8      1973502.07     13644039.51
      1973093.22     13644065.55      1972628.53     13644070.74
#Sta/Elev= 30
  3825.6  904.65    3898  902.52  3955.1  898.31  3960.3  898.89  3990.1  896.88
  3995.3  897.54  4030.3  895.13  4346.4  887.76    4577  879.79  4617.1  880.38
  4679.1  878.47  4743.5  874.19  4791.4  876.08  4800.5  875.46  4838.5  874.01
    4839  873.21  4845.3  874.01    5003  874.01    5010  874.01  5038.1  874.01
  5065.3  875.72  5235.7   876.5    5342  879.22  5446.1   884.9  5576.1  888.81
  5646.1  892.29  5716.1  892.63  5796.1  895.77  5833.6  898.93  5902.6  902.19
#Mann= 7 ,-1 , 0
  3825.6      .1       0  4800.5     .05       0  4838.5    .033       0
  4845.3     .05       0    5003      .1       0    5010     .05       0
    5342      .1       0
Bank Sta=4838.5,4845.3
XS Rating Curve= 0 ,0
Exp/Cntr=0.3,0.1

Type RM Length L Ch R = 1 ,215309  ,612,612,612
BEGIN DESCRIPTION:
Black Creek 231.0
END DESCRIPTION:
XS GIS Cut Line= 6
      1974520.33     13643604.61      1973551.55     13643792.11
      1973522.91     13643893.68       1973455.2      13643971.8
      1973338.01      13643971.8      1972625.05       13644025.
#Sta/Elev= 30
  3848.2  901.42  3965.7  895.64  4193.6  889.73  4536.1  878.48    4587  877.77
  4612.9  879.24    4618  878.34  4664.7  879.99  4709.2  880.22  4800.9  879.08
  4833.9  877.41  4848.3  876.06  4906.5  874.01    4907  873.21  4912.8  873.21
  4913.3  874.01  5128.8  874.01  5254.3  874.31  5270.3  874.65  5275.3  876.07
  5294.4   876.7  5334.5  877.52  5354.6  877.04  5394.7  878.54  5424.8  883.65
    5495  886.68  5645.4  895.14  5735.7  896.16  5785.8  898.64    5876  904.72
#Mann= 5 ,-1 , 0
  3848.2      .1       0  4833.9     .05       0  4906.5    .033       0
  4913.3     .05       0  5128.8      .1       0
Bank Sta=4906.5,4913.3
XS Rating Curve= 0 ,0
Exp/Cntr=0.3,0.1

Type RM Length L Ch R = 1 ,214697  ,50,50,50
BEGIN DESCRIPTION:
Mapping XS 2f5a4afb
END DESCRIPTION:
XS GIS Cut Line= 6
      1973991.69     13643266.06      1973384.89      13643596.8
      1973298.95     13643609.82       1973080.2     13643612.43
      1972884.89     13643612.43      1972572.36     13643672.33
#Sta/Elev= 30
  3889.1  899.87  3899.9  898.59  3953.7  897.13  3981.5  894.79  4025.2  892.98
  4166.7  889.34    4216  886.41  4248.3  885.77  4275.8  886.82  4313.8  886.37
  4439.1   882.5  4542.6  876.84  4653.7  874.25  4675.4  874.01    4676  873.21
  4682.1  873.21  4682.6  874.01  4876.7  874.01  5031.1  874.39  5041.1  875.52
  5051.1  878.78  5061.1  880.49  5083.7  882.13  5111.6  886.21  5182.9  889.49
  5195.5   891.2  5213.4  894.53  5233.8  897.13  5337.3  903.48  5399.4  904.44
#Mann= 6 ,-1 , 0
  3889.1      .1       0  4653.7     .05       0  4675.4     .07       0
  4682.6     .05       0  4876.7      .1       0  5195.5     .16       0
Bank Sta=4675.4,4682.6
XS Rating Curve= 0 ,0
Exp/Cntr=0.3,0.1

Type RM Length L Ch R = 1 ,214647  ,34,34,34
BEGIN DESCRIPTION:
Black Creek 230.0
END DESCRIPTION:
XS GIS Cut Line= 5
      1973926.55     13643268.68      1973317.18     13643575.97
      1972983.84     13643565.55      1972869.26     13643573.36
      1972564.55     13643638.47
#Sta/Elev= 30
  3943.8  898.81  4015.8  894.83  4105.1  891.55  4144.1  891.34  4261.2  885.98
  4382.3   884.6  4471.9  881.08  4500.9  877.79  4523.2  876.62  4586.6  875.44
  4587.1  874.64  4593.2  874.64  4593.8  875.44  4648.5  875.73  4674.8   877.4
  4808.5  876.33  4815.4   876.4  4820.4  878.71  4842.7   878.7  5038.8  879.87
  5089.2  882.49  5110.6  885.69  5140.3  888.01    5171  888.97  5202.1  892.99
  5211.9  894.29  5248.8  896.17  5253.9  897.32  5347.8  903.15  5386.2   903.4
#Mann= 6 ,-1 , 0
  3943.8      .1       0  4586.6     .07       0  4593.8      .1       0
  4674.8     .05       0  4842.7      .1       0  5202.1     .16       0
Bank Sta=4586.6,4593.8
XS Rating Curve= 0 ,0
Exp/Cntr=0.3,0.1

Type RM Length L Ch R = 1 ,214613  ,228,228,228
BEGIN DESCRIPTION:
Mapping XS b399f054
END DESCRIPTION:
XS GIS Cut Line= 5
      1973910.96     13643240.02       1973330.2     13643529.09
      1973116.66     13643526.49      1972884.89     13643539.51
       1972554.2     13643609.81
#Sta/Elev= 30
  3950.5  899.69  3967.8  899.89  4107.8  893.05  4191.7  891.92  4225.3  889.66
  4242.1  890.05  4247.7  888.76  4286.9  889.12  4292.5  888.03  4309.3   888.2
    4382  883.14  4437.5   882.8  4533.2  876.55    4722  873.06  4817.2  872.52
  4872.5  872.65  4877.5  876.28  4934.6  874.12  4964.7  870.57  5011.2  868.89
  5011.7  868.09  5018.4  868.89  5034.8  871.84  5042.4  875.27    5055  877.87
  5085.7  880.82  5106.1  884.01  5210.3  893.36  5341.3  901.89    5383  902.13
#Mann= 6 ,-1 , 0
  3950.5      .1       0    4722     .05       0  4817.2      .1       0
  5011.2     .07       0  5018.4      .1       0  5210.3     .16       0
Bank Sta=5011.2,5018.4
XS Rating Curve= 0 ,0
Exp/Cntr=0.3,0.1

Type RM Length L Ch R = 1 ,214385  ,414,414,414
BEGIN DESCRIPTION:
Black Creek 229.0
END DESCRIPTION:
XS GIS Cut Line= 3
      1973462.99     13643180.14        1972875.       13643325.
      1972489.54      13643422.2
#Sta/Elev= 30
  4410.7  895.08  4439.5  893.95  4480.7  891.03  4489.8  891.01  4536.4  887.68
  4542.5  886.68  4624.9  879.98  4707.6  874.32    4800   870.9  4933.9  869.66
  4951.4  868.61  4985.4  868.15  4992.9  866.82  5002.4  866.71  5002.9  865.91
  5009.1  865.91  5009.6  866.71  5013.7  867.52  5018.8  867.52  5034.2  871.73
  5047.2  873.33  5080.5  876.01  5116.4  880.19  5121.5  880.24  5150.3  884.22
  5222.5  890.25  5239.6  892.49  5274.1  895.45  5362.8  897.54  5413.8  898.03
#Mann= 3 ,-1 , 0
  4410.7      .1       0  5002.4     .07       0  5009.6      .1       0
Bank Sta=5002.4,5009.6
XS Rating Curve= 0 ,0
Exp/Cntr=0.3,0.1

Type RM Length L Ch R = 1 ,213971  ,386,386,386
BEGIN DESCRIPTION:
Black Creek 228.0
END DESCRIPTION:
XS GIS Cut Line= 3
      1973375.02     13642824.99      1972697.39     13643023.89
      1972423.97     13643286.89
#Sta/Elev= 30
  4562.3  900.51  4617.6  896.79  4635.3  894.57  4645.7  892.72    4651  890.89
  4666.5  889.21    4723  885.81  4756.4  882.03  4828.4  875.77  4895.1  872.48
  4924.7  872.13  4938.9  871.24  4958.4  865.88  4972.3  866.48    4986  865.72
  4986.5  864.92  4992.7  864.92  4993.3  865.72  5005.7  868.16  5010.9  866.92
  5039.1  869.76  5104.3  866.87  5156.4  867.12  5216.5  873.25  5249.8  874.62
  5267.2  876.58  5306.4  878.66  5419.6  886.97  5532.8   891.7  5647.9  894.86
#Mann= 4 ,-1 , 0
  4562.3      .1       0  4924.7     .16       0    4986     .07       0
  4993.3      .1       0
Bank Sta=4986,4993.3
XS Rating Curve= 0 ,0
Exp/Cntr=0.3,0.1

Type RM Length L Ch R = 1 ,213585  ,278,278,278
BEGIN DESCRIPTION:
Black Creek 227.0
END DESCRIPTION:
XS GIS Cut Line= 3
       1973319.8     13642581.17      1972689.57      13642721.8
      1972297.52     13643181.37
#Sta/Elev= 30
  4420.7  893.82  4461.4  891.38  4466.6  890.31  4509.9  886.85  4548.3  882.68
  4630.5  875.73  4688.9  872.39  4829.4  868.98  4886.7  866.84    4970  866.31
  4995.7  865.44  4996.3  864.64  5002.5  864.64    5003  865.44  5040.4  865.82
  5056.9  867.58  5062.1  866.55  5071.8  867.13  5079.2  866.37  5114.3   867.1
  5149.5  869.19  5284.5  872.97    5313  875.42  5327.3  878.34  5341.6  879.92
  5370.2  881.71  5419.6  883.23  5497.5  882.63  5624.9  891.16  5670.5   892.2
#Mann= 3 ,-1 , 0
  4420.7      .1       0  4995.7     .07       0    5003      .1       0
Bank Sta=4995.7,5003
XS Rating Curve= 0 ,0
Exp/Cntr=0.3,0.1

Type RM Length L Ch R = 1 ,213307  ,320,320,320
BEGIN DESCRIPTION:
Black Creek 226.0
END DESCRIPTION:
XS GIS Cut Line= 3
      1973374.96     13642524.99      1972710.41     13642435.34
      1971938.45     13642713.46
#Sta/Elev= 30
  4424.2  896.19  4474.6  893.49  4533.2   888.1  4605.8  883.43  4683.7  876.63
  4761.5  871.48  4767.2  870.55  4811.7  869.23  4888.3  868.35  4906.9  865.37
  4914.8  865.36  4915.4  864.56  4921.7  864.56  4922.3  865.36  5125.2  865.36
  5199.3  865.37  5217.4  867.66  5260.6  868.41  5280.7  870.31    5286  870.17
  5302.5  872.31  5334.4  874.25  5403.5  876.29  5515.1  877.39  5643.7  884.95
  5669.1   885.3  5694.5  884.65  5780.8  886.85    5812  888.31  5915.3  896.13
#Mann= 5 ,-1 , 0
  4424.2      .1       0  4811.7     .05       0  4914.8    .033       0
  4922.3     .05       0  5125.2      .1       0
Bank Sta=4914.8,4922.3
XS Rating Curve= 0 ,0
Exp/Cntr=0.3,0.1

Type RM Length L Ch R = 1 ,212987  ,633,633,633
BEGIN DESCRIPTION:
Black Creek 225.0
END DESCRIPTION:
XS GIS Cut Line= 3
      1973632.33     13642357.23      1972668.74     13642091.59
      1971874.45     13642070.76
#Sta/Elev= 30
  4286.6  897.51  4418.7  890.48    4512  880.73  4573.1  882.54  4691.8  876.78
  4781.7  877.41  4805.3  876.36  4895.8  867.17  4947.7  865.69  4953.2  866.94
  4968.4  867.61    4989  862.85  4989.6  862.05  4995.9  862.05  4996.5  862.85
  5009.9   865.6  5027.1  867.21  5032.3  866.24  5061.5  868.95  5106.2  870.31
  5238.1  868.54  5319.9  866.28  5345.9  867.94  5350.9  866.73  5389.9  870.42
  5459.9  873.42    5520  873.51    5570  869.98  5900.1  876.45  6080.7  881.22
#Mann= 3 ,-1 , 0
  4286.6      .1       0    4989     .07       0  4996.5      .1       0
Bank Sta=4989,4996.5
XS Rating Curve= 0 ,0
Exp/Cntr=0.3,0.1

Type RM Length L Ch R = 1 ,212354  ,216,216,216
BEGIN DESCRIPTION:
Black Creek 224.0
END DESCRIPTION:
XS GIS Cut Line= 3
      1973325.03     13641875.01      1972756.41     13641683.61
       1971964.7     13641551.66
#Sta/Elev= 30
  4459.8   880.5  4475.6  880.21  4554.8   875.9  4690.8   872.7  4713.1  870.98
  4722.3   871.3  4744.7  870.44  4765.8  868.51  4797.5  864.27  4881.7  861.03
  4912.7  860.13  4913.3  859.33  4919.8  859.33  4920.4  860.13  4992.6  860.13
  5050.7  860.14  5071.3  861.32  5139.9  863.11  5223.4  863.45  5327.4  864.82
  5449.1  867.64  5570.7  871.01  5578.2  871.83  5608.6  872.83  5639.1   875.1
  5699.9  877.54  5760.7  878.41    5781     880  5814.1  880.27  5862.4  881.66
#Mann= 5 ,-1 , 0
  4459.8      .1       0  4881.7     .05       0  4912.7     .07       0
  4920.4     .05       0  4992.6      .1       0
Bank Sta=4912.7,4920.4
XS Rating Curve= 0 ,0
Exp/Cntr=0.3,0.1

Type RM Length L Ch R = 1 ,212138  ,41,41,41
BEGIN DESCRIPTION:
Mapping XS b1644f6e
END DESCRIPTION:
XS GIS Cut Line= 6
      1973693.91     13641405.83      1973263.36     13641419.72
      1972975.16     13641513.47      1972850.16     13641499.58
      1972631.41     13641478.75      1971982.09     13641444.02
#Sta/Elev= 30
  4191.3  894.91  4290.3  884.51  4340.3  881.14  4373.1  877.89  4420.3  873.69
  4470.4  870.13  4500.4  869.18  4540.4  865.13  4560.4  864.16  4610.4  862.98
  4682.9  863.28    4831  861.68  4847.9  862.06  4907.9  860.12  4908.5  859.32
    4915  859.32  4915.6  860.12    5100  860.78  5151.7  860.78  5156.8  862.35
  5186.7  860.51  5226.9  861.83  5259.7  861.58  5287.1  863.01  5327.1  862.59
  5447.3   864.5  5622.1  870.54  5687.7  874.99  5757.8  877.94  5920.9  881.55
#Mann= 6 ,-1 , 0
  4191.3     .16       0  4373.1      .1       0    4831     .05       0
  4907.9    .033       0  4915.6     .05       0    5100      .1       0
Bank Sta=4907.9,4915.6
XS Rating Curve= 0 ,0
Exp/Cntr=0.3,0.1

Type RM Length L Ch R = 1 ,212097  ,46,46,46
BEGIN DESCRIPTION:
Mapping XS ee527b7d
END DESCRIPTION:
XS GIS Cut Line= 6
      1973693.95     13641381.52      1973256.41     13641374.58
      1972940.44     13641461.39       1972832.8      13641471.8
      1972735.58      13641471.8      1971982.13      13641409.3
#Sta/Elev= 30
  4197.7  891.98  4226.7  890.31  4306.7  882.24  4381.6  876.05  4446.7  870.11
  4496.7  868.76  4526.7  865.58  4556.7  863.78  4576.7  863.73  4616.7  865.93
  4709.8  867.46  4940.3  866.49  5053.3   865.1    5102  865.45    5139  865.18
  5171.3  863.01  5187.2  860.66  5192.2   861.9  5205.3  860.64  5205.9  859.84
  5212.4  859.84    5213  860.64  5289.5  863.05  5312.9  862.26  5359.7  862.83
  5510.2   866.2  5640.7  871.06  5690.8  874.52  5771.1  877.68  5924.5  881.35
#Mann= 6 ,-1 , 0
  4197.7     .16       0  4381.6      .1       0  4940.3     .05       0
    5102      .1       0  5205.3    .033       0    5213      .1       0
Bank Sta=5205.3,5213
XS Rating Curve= 0 ,0
Exp/Cntr=0.3,0.1

Type RM Length L Ch R = 1 ,212051  ,228,228,228
BEGIN DESCRIPTION:
Mapping XS d3e7b8dc
END DESCRIPTION:
XS GIS Cut Line= 6
      1973700.87     13641332.91      1973266.83     13641336.39
       1973020.3     13641395.41      1972839.75     13641433.61
      1972752.94     13641437.08      1971999.74     13641357.25
#Sta/Elev= 30
  4196.7  890.76  4202.6  889.13  4212.6  887.92  4367.1  876.67  4390.4  874.39
  4502.6  865.48  4532.6  864.19  4731.2  860.98  4905.7  859.59  4910.8  860.19
  4950.3  859.23  4955.4  859.86  4981.7  858.39  4996.2  856.55  4996.8  855.75
  5003.3  855.75  5003.9  856.55  5012.3  858.57  5032.8  859.21  5183.8  860.52
  5203.9  859.79  5254.2  860.96  5284.3  862.85  5318.6  862.03    5509   865.7
  5535.7  867.33  5636.3  870.82  5706.7  874.69  5817.3  878.77  5913.1   880.8
#Mann= 5 ,-1 , 0
  4196.7      .1       0  4367.1     .16       0  4390.4      .1       0
  4996.2     .07       0  5003.9      .1       0
Bank Sta=4996.2,5003.9
XS Rating Curve= 0 ,0
Exp/Cntr=0.3,0.1

Type RM Length L Ch R = 1 ,211823  ,433,433,433
BEGIN DESCRIPTION:
Mapping XS 90645dd4
END DESCRIPTION:
XS GIS Cut Line= 4
      1973792.93      13641291.6      1973290.32     13641150.97
      1972386.67     13641247.33       1971881.5      13641231.7
#Sta/Elev= 30
  4045.4  896.31  4055.1  894.76  4089.2   893.5  4115.9  891.33  4136.7  887.38
  4196.8  883.13  4241.3  877.96  4282.1  874.38  4365.2  868.88  4422.4  863.09
  4541.7  860.57  4723.5  858.91  4914.6  857.57  4954.8  858.38  4974.9  857.89
  4991.1  856.27  4991.8  855.47  4998.3  855.47  4998.9  856.27  5015.2  856.43
    5030  857.97  5045.3  857.49  5186.1  858.86  5276.6  861.69  5409.7  864.51
  5517.8  867.98  5627.8  873.22    5713  876.13  5837.9  879.73  5981.5  882.39
#Mann= 3 ,-1 , 0
  4045.4      .1       0  4991.1     .07       0  4998.9      .1       0
Bank Sta=4991.1,4998.9
XS Rating Curve= 0 ,0
Exp/Cntr=0.3,0.1

Type RM Length L Ch R = 1 ,211390  ,627,627,627
BEGIN DESCRIPTION:
Mapping XS d1661463
END DESCRIPTION:
XS GIS Cut Line= 4
      1973982.11     13641187.08      1973291.14     13640919.72
      1972423.08     13640739.16      1971975.79     13641030.42
#Sta/Elev= 30
  3672.9  903.61  3712.7  904.21  3749.1  902.34  3852.1  891.95  3882.7  886.23
    3918  883.79  3948.6   879.9  4184.5  862.15  4389.4  857.71    4493  857.03
  4508.8  859.34  4522.2  859.64  4532.4  859.17  4552.8  856.37  4569.4  855.87
    4570  855.07  4576.5  855.07  4577.2  855.87  4592.9  855.87  4692.8  855.87
  4838.8  855.87  4930.8  857.11  4971.6  855.87  5022.7  855.87  5032.9  856.39
  5049.5  859.43  5104.7  862.03    5469  871.42  5779.9  877.67  5834.2  879.53
#Mann= 6 ,-1 , 0
  3672.9      .1       0    4493     .16       0  4569.4     .07       0
  4577.2     .16       0  4592.9     .05       0  4692.8      .1       0
Bank Sta=4569.4,4577.2
XS Rating Curve= 0 ,0
Exp/Cntr=0.3,0.1

Type RM Length L Ch R = 1 ,210763  ,44,44,44
BEGIN DESCRIPTION:
Mapping XS 2f0ff378
END DESCRIPTION:
XS GIS Cut Line= 4
       1974016.8     13641034.29      1973419.61     13640680.14
      1972891.83     13640489.16      1972124.51     13640485.69
#Sta/Elev= 30
  4138.1  893.76  4161.9  894.02  4167.7  893.23  4183.3  894.14  4204.7  893.96
  4226.2  892.32  4241.8  892.57  4291.3  889.16  4306.1  887.82  4321.7  884.58
  4380.1   880.6    4386  879.08  4395.8  879.35    4423  876.83    4577  860.59
  4822.2  855.87  4822.8  855.07  4829.4  855.07    4830  855.87  4908.6  855.87
  4938.2  855.87  5190.4  855.96  5237.6  855.87  5332.1  855.89  5460.5  860.59
  5680.5   861.8  5890.5  864.87  5950.5  866.78  6070.5   874.3    6161  878.22
#Mann= 7 ,-1 , 0
  4138.1      .1       0  4822.2    .033       0    4830      .1       0
  4908.6     .16       0  4938.2     .05       0  5190.4     .16       0
  5237.6      .1       0
Bank Sta=4822.2,4830
XS Rating Curve= 0 ,0
Exp/Cntr=0.3,0.1

Type RM Length L Ch R = 1 ,210719  ,53,53,53
BEGIN DESCRIPTION:
Mapping XS 4ff97281
END DESCRIPTION:
XS GIS Cut Line= 4
      1974048.08     13641020.41      1973523.77     13640676.66
      1972905.72      13640447.5      1972118.73      13640447.5
#Sta/Elev= 30
  4124.1  890.86  4144.4  890.04  4159.5  891.52  4180.6  890.89  4195.7  891.77
    4268  889.69  4289.1  887.11  4304.2  887.28  4367.4  879.37  4433.8  874.63
  4548.3     863  4614.7  860.16  4769.4  856.64    4770  855.84  4777.2  856.64
  4828.7  860.35  4875.7  860.06  4966.8  859.64  5079.3  859.64  5239.6  859.58
  5313.2  859.44  5318.5  858.28  5343.6  858.36  5348.9   856.7  5379.3  856.88
  5480.9  860.02  5700.9  861.07  5940.9  864.77  6100.9  874.33  6197.2  878.46
#Mann= 7 ,-1 , 0
  4124.1      .1       0  4769.4    .033       0  4777.2      .1       0
  4875.7     .16       0  4966.8     .05       0  5079.3     .16       0
  5239.6      .1       0
Bank Sta=4769.4,4777.2
XS Rating Curve= 0 ,0
Exp/Cntr=0.3,0.1

Type RM Length L Ch R = 1 ,210666  ,373,373,373
BEGIN DESCRIPTION:
Mapping XS ff79defb
END DESCRIPTION:
XS GIS Cut Line= 4
      1974037.64     13640989.15      1973468.22     13640614.16
      1973044.61     13640423.19       1972145.3     13640398.89
#Sta/Elev= 30
  4161.2  888.42  4180.1  888.44  4195.2  890.17  4267.4  888.78  4375.9  879.73
  4427.1  876.58  4475.7  870.21  4562.6  862.51  4779.4  856.74    4787   855.6
  4898.8  854.76  4973.7  853.01  4979.2  851.76  4998.4  851.27    4999  850.47
  5006.3  851.27  5172.2  853.81  5192.9  857.16  5198.4  854.54    5216  857.32
  5221.5   854.6  5238.3  854.75  5367.3  856.14  5487.3  860.05  5677.4  860.29
  5897.5  862.41  5977.5  864.66  6037.5  868.08  6057.5   870.5  6207.3  877.41
#Mann= 5 ,-1 , 0
  4161.2      .1       0  4998.4     .07       0  5006.3      .1       0
  5172.2     .16       0  5238.3      .1       0
Bank Sta=4998.4,5006.3
XS Rating Curve= 0 ,0
Exp/Cntr=0.3,0.1

Type RM Length L Ch R = 1 ,210293  ,514,514,514
BEGIN DESCRIPTION:
Mapping XS c7e4763e
END DESCRIPTION:
XS GIS Cut Line= 4
       1974419.6     13640652.35      1973881.41     13640350.27
      1972884.89     13640065.55      1972065.45     13640336.38
#Sta/Elev= 30
  4005.6  887.89  4009.8  887.75    4086   885.7  4116.2  884.32  4169.8  885.05
  4213.1  883.97  4218.9  882.71  4272.5  880.33  4353.4  872.72  4359.2  873.72
  4375.1  870.84  4418.5  867.78  4558.8     862  4769.6  855.92  4785.4  854.49
  4899.8  852.78  5010.3  849.11  5010.9  848.31  5018.2  849.11    5087   854.9
  5099.8  852.09  5107.8  851.73  5245.4  853.12  5668.8  853.64  6048.7  857.85
  6206.7  861.55    6277  867.66  6354.2  872.47  6467.4  878.09  6522.2  879.47
#Mann= 5 ,-1 , 0
  4005.6      .1       0  4009.8     .16       0    4086      .1       0
  5010.3     .07       0  5018.2      .1       0
Bank Sta=5010.3,5018.2
XS Rating Curve= 0 ,0
Exp/Cntr=0.3,0.1

Type RM Length L Ch R = 1 ,209779  ,682,682,682
BEGIN DESCRIPTION:
Mapping XS 9cff2789
END DESCRIPTION:
XS GIS Cut Line= 4
      1974822.36     13639450.99      1974110.58     13639891.94
       1973207.8     13639916.25      1972371.03      13640058.6
#Sta/Elev= 30
  3832.8  890.72  3885.3  885.88  4029.7   878.1  4080.2  878.17  4174.7  874.46
  4335.5     877  4421.7  874.81  4488.4  870.01  4568.2  860.36  4582.6  861.07
  4589.4  858.46  4595.3  859.95  4617.8  856.86  4647.3   855.4 4781.02  851.71
  4815.2  851.25  4875.8  850.48  4935.8  846.65  4970.2  848.49  4991.6  845.89
  4992.3  845.09  4999.9  845.89  5005.8  848.44  5025.8  850.91  5205.9  850.84
  5225.9  849.41  5355.9     851 5777.59  851.71  6256.1  855.66    6422   858.8
#Mann= 4 ,-1 , 0
  3832.8      .1       0  4815.2     .16       0  4991.6     .07       0
  4999.9      .1       0
Bank Sta=4781.02,5777.59
XS Rating Curve= 0 ,0
Exp/Cntr=0.3,0.1

Type RM Length L Ch R = 1 ,209097  ,313,313,313
BEGIN DESCRIPTION:
Mapping XS f923c0cc
END DESCRIPTION:
XS GIS Cut Line= 4
      1974523.75     13639530.83      1974002.94     13639537.77
      1973416.14     13639735.69      1972569.41     13639822.45
#Sta/Elev= 30
  4006.5  875.38  4065.3   873.3  4175.3  871.89  4226.8  871.34  4385.3   868.9
  4532.4  864.73  4620.2  857.53  4651.8   853.1  4658.3  851.58  4689.8  849.96
 4742.83   849.6  4784.2  849.43  4862.9  847.76    4884  848.37  4903.6   847.1
    4973  846.36  4993.7  843.27  4995.1  843.02  4995.8  842.22  5002.7  842.22
  5003.4  843.02  5021.2  846.61  5030.7  849.83  5052.9  850.29    5074  848.38
 5105.48   849.6  5424.4  849.96  5690.4  850.34  5861.5  851.08  5997.8  852.94
#Mann= 9 ,-1 , 0
  4006.5      .1       0  4175.3     .16       0  4226.8      .1       0
  4903.6     .16       0  4993.7      .1       0  4995.1     .07       0
  5003.4      .1       0  5424.4     .05       0  5690.4      .1       0
Bank Sta=4742.83,5105.48
XS Rating Curve= 0 ,0
Exp/Cntr=0.3,0.1

Type RM Length L Ch R = 1 ,208784  ,465,465,465
BEGIN DESCRIPTION:
Black Creek 220.0
END DESCRIPTION:
XS GIS Cut Line= 3
      1974429.99     13639398.89      1973537.66      13639447.5
      1972334.55     13639583.27
#Sta/Elev= 30
  4249.7  871.77  4438.1   867.8    4457  868.08  4525.1  865.07  4625.4  863.98
  4731.4  860.76  4745.4   860.3  4805.5  848.93  4855.6  847.86  4935.7  848.31
  4975.8  843.49  4981.6  840.39  4982.3  839.59  4989.2  839.59  4989.9  840.39
  5025.8  845.29  5035.9   847.9  5055.9  850.81  5065.9  850.46  5075.9  848.87
  5085.9  849.57  5126.3  849.01  5253.3   848.7  5276.9  846.87  5417.7  848.64
    5433  847.91  5679.4  847.17  5920.9  847.72    6147  850.17  6354.1     855
#Mann= 7 ,-1 , 0
  4249.7      .1       0  4438.1     .16       0  4625.4      .1       0
  4731.4     .16       0  4981.6     .07       0  4989.9     .16       0
  5126.3      .1       0
Bank Sta=4981.6,4989.9
XS Rating Curve= 0 ,0
Exp/Cntr=0.3,0.1
