HEC-RAS study Black Creek.prj: Black Creek Base Level Engineering

--- Black Creek.g01 (geometry) --- (continued)

Type RM Length L Ch R = 1 ,177331  ,799,799,799
BEGIN DESCRIPTION:
Mapping XS c044850c
END DESCRIPTION:
XS GIS Cut Line= 3
      1974785.18     13619104.39      1974056.04     13618868.29
      1971369.31      13618722.5
#Sta/Elev= 30
    3998  771.09  4173.1  765.38  4338.3  761.89  4466.3  757.02 4549.26  755.51
  4626.3  754.81  4670.9  753.28  4681.4  754.39  4722.3  754.83  4955.7  755.13
  4965.7   754.8  4985.8  750.56  4988.7  746.86  4989.7  746.06  5001.9  746.06
  5002.8  746.86  5005.8  748.62  5025.8  753.87  5035.9  755.36    5043  755.12
  5086.5  754.94  5284.2  755.29  5506.5  755.27    5847   753.6 6156.75  755.51
  6447.9   755.6  6846.1  757.45  7088.9  759.51  7369.3  765.33  7455.1  765.65
#Mann= 7 ,-1 , 0
    3998      .1       0  4988.7     .07       0  5002.8      .1       0
    5043     .05       0  5086.5      .1       0  5284.2     .05       0
  6846.1      .1       0
Bank Sta=4549.26,6156.75
XS Rating Curve= 0 ,0
Exp/Cntr=0.3,0.1

Type RM Length L Ch R = 1 ,176532  ,1113,1113,1113
BEGIN DESCRIPTION:
Black Creek 179.0
END DESCRIPTION:
XS GIS Cut Line= 4
      1974993.85     13618871.59      1974370.62     13618338.63
      1972500.83     13617954.95      1971702.23     13618454.94
#Sta/Elev= 30
  3676.9  772.21    3830  773.42    4021  770.28  4092.3  770.57  4227.4   768.5
    4369     764  4544.2  760.13 4746.17  753.07  4849.8  751.12  4891.9  752.67
    4911  751.44  4921.2  749.62  4942.3  753.14  4951.8  750.44  4962.1  750.09
  4972.3  753.83  4982.5  752.82  4985.6  746.83  4986.6  746.03  4998.8  746.03
  4999.7  746.83  5013.1  751.93  5023.3  753.78  5098.6  754.28  5207.1   752.8
    5646  752.03  5850.2  750.67 6542.43  753.07  6986.1  755.64  7347.9   759.5
#Mann= 5 ,-1 , 0
  3676.9      .1       0  4985.6     .07       0  4999.7      .1       0
  5098.6     .05       0  6986.1      .1       0
Bank Sta=4746.17,6542.43
XS Rating Curve= 0 ,0
Exp/Cntr=0.3,0.1

Type RM Length L Ch R = 1 ,175419  ,147,147,147
BEGIN DESCRIPTION:
Black Creek 177.0
END DESCRIPTION:
XS GIS Cut Line= 5
      1974718.74     13618593.44      1973805.52      13617631.6
      1973154.47      13617506.6      1972623.96     13617505.21
      1971651.45     13617600.13
#Sta/Elev= 30
  3487.6  769.58  3736.6  766.35  3835.7  763.64  3849.9  763.88  3878.2  762.81
    4345  753.99  4649.1  751.43  4797.6  751.97  4924.9  751.24    4957  749.84
  4967.2  748.13  4969.6  745.78  4970.7  744.98    4983  744.98  4984.1  745.78
  4990.6  746.12  5008.7  746.29  5028.3   747.5    5034   748.4    5039  750.54
  5048.6  751.18  5079.2  750.22  5099.6  750.94  5168.8   750.6  5402.9  749.27
  5626.3  749.06  5963.6  752.22  6572.7   757.2  6781.1  760.83  6984.5  767.43
#Mann= 7 ,-1 , 0
  3487.6      .1       0  4969.6     .03       0  4984.1      .1       0
  4990.6     .05       0  5008.7      .1       0  5168.8     .05       0
  5963.6      .1       0
Bank Sta=4969.6,4984.1
XS Rating Curve= 0 ,0
Exp/Cntr=0.3,0.1

Type RM Length L Ch R = 1 ,175272  ,1454,1454,1454
BEGIN DESCRIPTION:
Mapping XS 5c1106e2
END DESCRIPTION:
XS GIS Cut Line= 6
       1974769.9     13618548.24      1974105.86     13617684.55
      1973858.47     13617545.66      1973372.36     13617411.11
      1972608.47     13617367.71      1971698.52     13617567.03
#Sta/Elev= 30
  3349.1  768.32  3696.8  763.55  4203.3  754.34  4658.1  750.93  4764.3  751.15
  4974.9  751.07  4988.4   745.2  4989.5   744.4  5001.8   744.4  5002.9   745.2
  5003.4  747.39  5008.6   747.5  5016.4  751.03  5156.2  751.26  5213.5  749.86
  5414.3  748.68  5444.4  749.34  5574.6  747.91  5604.6  749.06  5654.7  749.02
  5744.8  753.32  5804.9  754.59    5835  754.12  5905.1  755.66  6006.6  755.61
  6138.1  757.39  6377.8   756.7  6519.5  757.68    6798  761.45  6923.3  766.07
#Mann= 5 ,-1 , 0
  3349.1      .1       0  4658.1     .05       0  4764.3      .1       0
  4988.4     .07       0  5002.9      .1       0
Bank Sta=4988.4,5002.9
XS Rating Curve= 0 ,0
Exp/Cntr=0.3,0.1

Type RM Length L Ch R = 1 ,173818  ,924,924,924
BEGIN DESCRIPTION:
Black Creek 172.0
END DESCRIPTION:
XS GIS Cut Line= 3
      1975562.06      13615950.6      1973704.39     13616523.52
      1972178.29     13616896.38
#Sta/Elev= 30
  3084.3  787.66  3285.6  778.66  3356.1  777.12  3646.3  766.17  3899.7  759.16
    4063   752.3  4378.9  747.76  4619.5  746.42  4874.1   747.6  4933.5   749.3
  4964.9  748.99  4973.9  742.75  4975.3  741.95  4989.1  742.75  5010.5  747.43
  5025.4  748.86  5120.3   749.2  5192.4  747.56  5470.3  746.57  5512.5  747.61
  5552.7   747.7  5583.6  744.46  5606.7  744.41    5635  744.93  5642.8  746.23
    5648  745.26  5665.9  748.34  5954.2  749.18  6304.2  756.45  6599.3  757.69
#Mann= 7 ,-1 , 0
  3084.3      .1       0  4874.1     .16       0  4973.9     .07       0
  4989.1     .16       0  5010.5      .1       0  5512.5     .16       0
  5606.7      .1       0
Bank Sta=4973.9,4989.1
XS Rating Curve= 0 ,0
Exp/Cntr=0.3,0.1

Type RM Length L Ch R = 1 ,172894  ,721,721,721
BEGIN DESCRIPTION:
Mapping XS 776d41fc
END DESCRIPTION:
XS GIS Cut Line= 3
      1975398.85     13615360.33      1973204.39     13615922.83
      1972023.83     13616582.56
#Sta/Elev= 30
  3092.2  783.02  3436.8  770.14  3773.9  754.37  3829.1  753.22  3849.8  754.17
  3942.7   750.6  4305.8  743.72  4359.2  743.18  4610.6  744.59  4675.6   744.6
  4706.8  745.97  4716.9  745.01  4892.4  745.92  4964.7  747.25    4975   746.9
    4982  742.35  4987.1  742.71  4988.1  741.54  4989.5  740.74  5003.3  741.54
    5006  743.93  5016.1  746.99  5376.6  744.65  5425.6   744.9    5463  742.19
  5519.4  745.94  6130.5  746.99  6292.7  748.28  6379.5   750.8    6710   752.6
#Mann= 9 ,-1 , 0
  3092.2      .1       0  4305.8     .16       0  4359.2      .1       0
  4610.6     .16       0  4988.1     .07       0  5003.3     .16       0
  5016.1      .1       0  5376.6     .16       0    5463      .1       0
Bank Sta=4988.1,5003.3
XS Rating Curve= 0 ,0
Exp/Cntr=0.3,0.1

Type RM Length L Ch R = 1 ,172173  ,675,675,675
BEGIN DESCRIPTION:
Mapping XS 9c67c889
END DESCRIPTION:
XS GIS Cut Line= 4
      1975093.29     13614770.05      1974141.89     13614929.77
      1972586.33     13615624.22      1971844.25     13616400.98
#Sta/Elev= 30
  3201.8  768.83  3281.2   767.1  3392.7  766.55    3484  763.51  3514.4  761.11
  3534.7  761.73  3585.4  759.16  3838.9  752.73  3889.6  750.54  4237.5  744.76
  4272.6  745.11  4387.7  742.06  4462.8  742.21  4502.6  740.11  4509.3  741.33
    4538  742.17  4865.4  744.34  4977.8  745.28  4984.4  744.81  4987.7  739.73
  4989.1  738.93    5003  739.73  5006.5  742.88  5017.3  745.39  5121.1  745.23
  5226.4  743.64  5637.5  742.11  5772.9  742.59  6246.3  745.53  6944.3  752.65
#Mann= 5 ,-1 , 0
  3201.8      .1       0  4865.4     .16       0  4987.7     .07       0
    5003     .16       0  5121.1      .1       0
Bank Sta=4987.7,5003
XS Rating Curve= 0 ,0
Exp/Cntr=0.3,0.1

Type RM Length L Ch R = 1 ,171498  ,56,56,56
BEGIN DESCRIPTION:
Mapping XS 6e2096c5
END DESCRIPTION:
XS GIS Cut Line= 6
       1974986.1      13614608.5      1973171.84      13614790.8
      1973119.75     13614730.04      1973058.99     13614756.08
      1973054.98     13615032.86      1971856.76     13616284.53
#Sta/Elev= 30
  3080.2   765.7    3196  764.51    3614  754.88  3792.6  747.72  4005.9  743.08
  4298.9  740.53  4317.5  741.69    4820  741.92  4850.2  739.89  4895.5  743.14
  4899.6  741.97  4919.8  742.41  4926.4  739.78  4947.3  736.28  4948.7  735.48
  4962.6  736.28  5005.1  739.74  5012.5  737.93  5030.6  739.91    5036  738.05
  5049.2  741.21  5078.7  738.58  5128.7  738.67  5265.6  744.84  5281.3  744.55
  5405.9  742.62  5576.6  742.48  5765.4  742.56  6445.6  745.25  7059.3  751.99
#Mann= 7 ,-1 , 0
  3080.2      .1       0  4947.3     .07       0  4962.6      .1       0
  5265.6     .12       0  5281.3      .1       0  5576.6     .12       0
  5765.4      .1       0
Bank Sta=4947.3,4962.6
XS Rating Curve= 0 ,0
Exp/Cntr=0.3,0.1

Type RM Length L Ch R = 1 ,171442  ,26,26,26
BEGIN DESCRIPTION:
Mapping XS a51ab042
END DESCRIPTION:
XS GIS Cut Line= 6
      1974996.01     13614582.56      1973196.42     13614759.93
      1973127.41     13614672.69      1973040.17     13614710.45
      1973029.76     13614979.98      1971746.05      13616214.5
#Sta/Elev= 30
  3046.6   765.7  3469.6  757.43  3670.6  752.38  3937.5  743.81  4253.4  741.39
  4273.5  740.36  4293.6  741.37  4625.2  741.24  4635.3  740.34  4645.3  741.37
  4775.9   741.6  4798.4   739.9  4799.8   739.1  4813.7   739.9  4826.2  740.16
  4853.1  744.81  4886.2  745.94  5336.7  746.42  5388.8  743.57  5432.4  742.97
  5598.9  742.37  5785.4  742.19    6280  743.94  6350.7  744.61  6357.9  745.71
  6372.1  744.59  6407.3  744.67    6485  746.22  6867.1  749.09  7134.7  753.91
#Mann= 7 ,-1 , 0
  3046.6      .1       0  4798.4     .07       0  4813.7      .1       0
  5336.7     .12       0  5432.4      .1       0  5598.9     .12       0
  5785.4      .1       0
Bank Sta=4798.4,4813.7
XS Rating Curve= 0 ,0
Exp/Cntr=0.3,0.1

Type RM Length L Ch R = 1 ,171416  ,295,295,295
BEGIN DESCRIPTION:
Mapping XS cd27af43
END DESCRIPTION:
XS GIS Cut Line= 6
      1974973.08     13614556.42      1973294.08     13614727.38
      1973163.16     13614643.23      1973011.25     13614677.95
      1972958.14     13614972.17      1971909.38     13615988.17
#Sta/Elev= 30
  3103.7  765.03  3704.9  752.51  3795.3  748.43  3966.2     744    4308  740.24
  4428.6   741.6  4639.7  740.33  4740.2  741.43  4780.4  740.13  4814.4  740.79
  4820.8  743.12  4835.2  739.82  4857.4  738.96  4858.8  738.16  4872.7  738.96
  4909.2  742.73  4974.5  743.31  4979.6  744.99  5022.6  742.02  5027.7  743.65
  5065.6  740.45  5070.7  741.98  5103.3  740.92  5161.2  742.94  5376.8  743.43
  5408.7  743.15  5653.4  741.93  5775.2  741.86  6338.9   744.2  6868.4  749.92
#Mann= 7 ,-1 , 0
  3103.7      .1       0  4857.4     .07       0  4872.7      .1       0
  5376.8     .12       0  5408.7      .1       0  5653.4     .12       0
  5775.2      .1       0
Bank Sta=4857.4,4872.7
XS Rating Curve= 0 ,0
Exp/Cntr=0.3,0.1

Type RM Length L Ch R = 1 ,171121  ,293,293,293
BEGIN DESCRIPTION:
Mapping XS a29bc30a
END DESCRIPTION:
XS GIS Cut Line= 2
      1975107.15     13614395.05      1970614.15     13614388.11
#Sta/Elev= 30
  2885.6   768.1  3207.7  759.06  3227.7  759.72  3560.3  752.99  3827.8  747.17
  3897.8   747.5  4207.8  740.54  4627.8  739.81  4667.8  738.19  4687.8  739.94
  4737.8   739.2  4757.8  737.45  4810.8  738.67  4837.8  739.54  4927.8  736.81
  4957.8  737.71  4977.8  736.55  4980.1  735.12  4981.5  734.32  4995.4  735.12
  5027.8  738.81  5101.2  738.65  5187.8  737.91  5387.8  740.05  5737.8  738.69
  6697.8  742.68  6767.8  744.56  6787.8  743.15  6895.8  743.76  7378.6  745.17
#Mann= 7 ,-1 , 0
  2885.6     .05       0  3560.3      .1       0  4810.8     .12       0
  4980.1     .07       0  4995.4     .12       0  5101.2      .1       0
  6895.8     .05       0
Bank Sta=4980.1,4995.4
XS Rating Curve= 0 ,0
Exp/Cntr=0.3,0.1

Type RM Length L Ch R = 1 ,170828  ,707,707,707
BEGIN DESCRIPTION:
Mapping XS c7ebeadb
END DESCRIPTION:
XS GIS Cut Line= 3
      1975114.07     13614186.72      1970814.89     13614166.08
      1970313.19      13614203.2
#Sta/Elev= 30
  2736.7  766.99  2945.8  762.36  2965.8     760  3925.8  743.04  3945.8  741.13
  4005.8  741.05  4045.8  745.73  4075.8  741.74  4295.8  741.33  4555.8  736.43
  4965.8  738.28  4985.8  734.44  4988.1  731.63  4989.5  730.83  5003.4  731.63
  5005.8  733.91  5015.8  736.22  5035.8   737.7  5275.8  738.62  5315.8  736.52
    5386  738.68  5390.5  738.63  5515.8  738.09  5565.8  734.95  5605.8  737.68
  5655.8  732.44  5675.8  736.22  5705.8  737.97  6995.8  741.04    7539  745.94
#Mann= 5 ,-1 , 0
  2736.7      .1       0  4988.1     .07       0  5003.4      .1       0
    5386     .05       0  5390.5      .1       0
Bank Sta=4988.1,5003.4
XS Rating Curve= 0 ,0
Exp/Cntr=0.3,0.1

Type RM Length L Ch R = 1 ,170121  ,1048,1048,1048
BEGIN DESCRIPTION:
Black Creek 171.0
END DESCRIPTION:
XS GIS Cut Line= 3
      1973886.65     13613381.17      1972280.78     13613641.58
      1970319.53     13614032.09
#Sta/Elev= 30
    3748  746.18  4043.5  746.92  4235.7  746.02  4448.7  742.94  4677.2  736.23
  4743.9  735.86  4762.7  733.97  4772.9  734.12  4793.1  736.63  4955.2   735.6
  4975.5  734.99  4985.3  732.91  4988.1  729.81  4989.5  729.01    5002  729.01
  5003.4  729.81  5005.9  732.12    5016  735.47  5026.1  736.15  5257.3   735.3
  5517.7  735.78  5615.3  735.78    5656  734.47  5677.8  735.84  5717.2  730.68
  5737.6   735.7  6298.4  738.01  6655.3  738.39    6853  739.65  7374.6  745.42
#Mann= 5 ,-1 , 0
    3748      .1       0  4988.1     .07       0  5003.4      .1       0
  5257.3     .05       0  5517.7      .1       0
Bank Sta=4988.1,5003.4
XS Rating Curve= 0 ,0
Exp/Cntr=0.3,0.1

Type RM Length L Ch R = 1 ,169073  ,602,602,602
BEGIN DESCRIPTION:
Black Creek 170.0
END DESCRIPTION:
XS GIS Cut Line= 3
      1973235.67     13612530.46      1972879.74     13612582.55
      1970171.36     13613546.11
#Sta/Elev= 30
  4259.3  743.94  4395.3  745.21    4605  741.43  4921.2  733.92  4963.7  732.71
  4969.2  731.34  4974.5  732.31  4984.9  728.99  4986.8  726.76  4988.4  725.96
  5002.6  726.76  5006.2  730.16  5025.6  733.52  5098.3  733.57  5621.1  732.55
  5682.8  730.47  5688.1  729.45  5738.5   732.6    5770  730.56    5781  731.47
  5800.8  728.89  5823.4  729.52  5831.7  731.02    5837   728.8  5844.7  731.92
  5855.3  733.16  6036.5  733.49  6401.7  734.48  6895.4  741.95  7493.7  746.12
#Mann= 5 ,-1 , 0
  4259.3      .1       0  4986.8     .07       0  5002.6      .1       0
  5098.3     .05       0  6036.5      .1       0
Bank Sta=4986.8,5002.6
XS Rating Curve= 0 ,0
Exp/Cntr=0.3,0.1

Type RM Length L Ch R = 1 ,168471  ,792,792,792
BEGIN DESCRIPTION:
Black Creek 169.0
END DESCRIPTION:
XS GIS Cut Line= 3
      1973452.67     13612009.63      1972845.01      13612070.4
      1969763.41     13612808.25
#Sta/Elev= 30
  4014.8  742.41  4123.5  739.86  4404.4  740.01  4535.1  741.59  4879.4  731.97
  4933.5  731.81  4968.7  731.47  4985.4  727.31  4995.7   726.6  5005.6  730.98
  5016.2  731.78  5035.4   731.4  5399.3  732.19  5651.5  731.18  5746.3   732.1
  5866.2  731.61  6040.2  730.77  6054.8  728.19  6057.2  726.49  6058.8  725.69
  6071.4  725.69    6073  726.49  6075.4  729.01  6082.2  730.73  6095.9   731.1
  6297.5  731.31  6554.9  735.58  6805.4  736.75  7248.1  743.95  7794.2  747.77
#Mann= 6 ,-1 , 0
  4014.8      .1       0  4933.5     .12       0  5035.4     .05       0
  5866.2      .1       0  6057.2     .07       0    6073      .1       0
Bank Sta=6057.2,6073
XS Rating Curve= 0 ,0
Exp/Cntr=0.3,0.1

Type RM Length L Ch R = 1 ,167679  ,747,747,747
BEGIN DESCRIPTION:
Black Creek 168.0
END DESCRIPTION:
XS GIS Cut Line= 3
      1973168.36     13611443.58        1972275.       13611475.
      1970133.65     13611714.41
#Sta/Elev= 30
  4121.9   741.8  4415.4  739.25  4525.5  736.81  4545.5  736.83  4655.6  733.42
  4675.6  733.31  4735.6  731.01  4872.1  728.34  4975.8  728.87  4985.8  728.28
  4987.9  724.36  4989.5  723.56  5002.1  723.56  5003.7  724.36  5005.8  726.84
  5013.3  728.41  5035.9  727.33  5059.5  727.84  5176.8  729.48  5307.6  730.46
  5627.6  729.48  5783.2  727.78  5790.6  725.66  5810.7  727.95  5921.4  729.61
  6042.2  730.23  6313.8  729.42    6681  735.08  6897.5  739.03  7170.5  739.74
#Mann= 5 ,-1 , 0
  4121.9      .1       0  4987.9     .07       0  5003.7      .1       0
  5059.5     .05       0  5627.6      .1       0
Bank Sta=4987.9,5003.7
XS Rating Curve= 0 ,0
Exp/Cntr=0.3,0.1

Type RM Length L Ch R = 1 ,166932  ,697,697,697
BEGIN DESCRIPTION:
Black Creek 166.0
END DESCRIPTION:
XS GIS Cut Line= 3
      1973140.64     13610846.36      1971800.31     13610769.97
      1970182.25     13611006.08
#Sta/Elev= 30
  4158.8  737.53  4541.1  732.63  4739.8  729.91  4926.7  725.72  4977.1  726.03
  4985.8  724.84  4987.8  722.56  4989.5  721.76  5002.1  721.76  5003.7  722.56
  5005.8  724.33  5015.8  724.92  5055.7  724.74  5075.9  725.63  5145.1  726.07
  5375.1  726.58  5720.7  727.81  5916.5  727.25  5921.6  724.12  5931.1  722.95
  5951.3  724.05  5961.4  725.72  5991.8  726.57  6092.8  727.95  6325.2  728.19
  6446.5  732.41  6527.4  732.67  6931.6  741.34  7026.4  741.17  7136.5  739.36
#Mann= 9 ,-1 , 0
  4158.8      .1       0  4541.1     .05       0  4739.8      .1       0
  4926.7     .12       0  4987.8     .07       0  5003.7     .12       0
  5055.7      .1       0  5375.1     .05       0  5720.7      .1       0
Bank Sta=4987.8,5003.7
XS Rating Curve= 0 ,0
Exp/Cntr=0.3,0.1

Type RM Length L Ch R = 1 ,166235  ,1025,1025,1025
BEGIN DESCRIPTION:
Black Creek 165.0
END DESCRIPTION:
XS GIS Cut Line= 3
      1973289.93     13610782.14      1971718.71     13609974.83
      1970190.94     13610269.96
#Sta/Elev= 30
  3858.7  738.78  3971.9  738.78  4016.3  737.47  4149.4  736.89  4505.1   728.1
    4654   725.9  4887.2  724.43  4975.5  724.19  4980.5  721.72  4982.2  720.92
  4994.8  720.92  4996.5  721.72  4997.7   722.8    5011  724.56  5066.2  724.58
  5142.5  724.52  5561.9  724.54  5908.7  725.69  5995.6  726.28  6066.9  724.47
  6078.2  722.33    6130  725.55  6168.8  724.52  6270.6  725.72  6596.4  726.46
  6688.2  727.45  6718.7  729.13    6757  728.37  6932.6  730.38  7181.2  736.25
#Mann= 7 ,-1 , 0
  3858.7      .1       0  4887.2     .12       0  4980.5     .07       0
  4996.5     .12       0  5066.2      .1       0  5142.5     .05       0
  5908.7      .1       0
Bank Sta=4980.5,4996.5
XS Rating Curve= 0 ,0
Exp/Cntr=0.3,0.1

Type RM Length L Ch R = 1 ,165210  ,714,714,714
BEGIN DESCRIPTION:
Black Creek 164.0
END DESCRIPTION:
XS GIS Cut Line= 4
      1973446.13      13610426.2       1972545.1     13609042.54
      1971237.81     13608813.37      1969809.53     13609757.45
#Sta/Elev= 30
  3997.6  732.98  4085.3  734.61  4106.4  732.75  4130.3  732.49  4321.5  732.82
  4541.1  733.67  4786.5  725.93  4966.7  721.13  5048.3  720.49  5096.8  721.66
  5256.5  722.42  5614.1  721.02  5742.4  719.92  5744.1  719.12  5758.4  719.92
  5762.2  720.09  6197.1  720.22  6887.5   722.7  7015.3  721.84    7095  722.59
  7186.7  721.17  7229.1  721.53  7347.9  723.78  7564.5  725.07  7895.6  729.84
  8043.1  730.14  8256.7  730.54  8292.9  731.66  8386.1  730.35  8688.1  732.39
#Mann= 11 ,-1 , 0
  3997.6      .1       0  4321.5     .05       0  4786.5      .1       0
  5096.8     .05       0  5614.1      .1       0  5742.4     .07       0
  5758.4      .1       0  5762.2     .05       0  7186.7      .1       0
  7229.1     .05       0  8043.1      .1       0
Bank Sta=5742.4,5758.4
XS Rating Curve= 0 ,0
Exp/Cntr=0.3,0.1

Type RM Length L Ch R = 1 ,164496  ,1370,1370,1370
BEGIN DESCRIPTION:
Mapping XS fe954851
END DESCRIPTION:
XS GIS Cut Line= 4
       1974071.3     13609733.38      1972105.99     13607913.91
      1970737.93      13607740.3        1968200.       13607650.
#Sta/Elev= 30
    4123  723.17  4453.2   720.8    4592  720.57  4890.7  720.22  4982.5  717.95
  5024.1  719.46  5626.6  718.65  5916.8  719.53  6195.9  718.12  6532.1  718.24
  6744.7  716.83  7202.3  717.74    7780  718.33  8119.9  717.33  8235.2  716.49
  8236.9  715.69  8251.2  716.49  8613.5  718.66  9083.8  719.16  9153.8  718.54
  9203.8  716.66  9233.9  718.11  9381.8  719.91    9504  721.62  9684.1   720.7
  9904.3   721.8  9994.3  723.35 10194.5  728.73 10460.8  741.06 10719.8  755.37
#Mann= 11 ,-1 , 0
    4123      .1       0  4453.2     .05       0    4592      .1       0
  5024.1     .05       0  6195.9      .1       0  7202.3     .05       0
  8119.9      .1       0  8235.2     .07       0  8251.2      .1       0
  9381.8     .05       0 10460.8      .1       0
Bank Sta=8235.2,8251.2
XS Rating Curve= 0 ,0
Exp/Cntr=0.3,0.1

Type RM Length L Ch R = 1 ,163126  ,976,976,976
BEGIN DESCRIPTION:
Black Creek 161.0
END DESCRIPTION:
XS GIS Cut Line= 4
      1975143.17     13610248.51      1974015.59     13608087.96
      1971598.92     13606831.02      1968659.37     13606407.49
#Sta/Elev= 30
  2104.5  739.44  2173.3  737.56  2201.1  738.61  2239.6  735.95  2394.2  733.95
  2758.4   724.2  2973.6  720.91  3284.9   718.9  3394.7   717.1  3501.8  716.83
  4094.6  716.78    4693  715.03  4782.6  714.87    4921  714.85  4967.8  713.21
  5967.8  713.36  6293.8  715.28  7028.5  715.11  7761.1  717.78  8181.1  712.31
  8182.9  711.51  8197.2  712.31  8355.7  713.62  8381.6  713.73  8441.5  713.99
  8465.8  712.35    8583   715.1  9311.8  719.87  9410.7  721.74 10235.5  726.82
#Mann= 15 ,-1 , 0
  2104.5      .1       0  3284.9     .05       0  3394.7      .1       0
  3501.8     .05       0  4094.6      .1       0    4693     .05       0
  4782.6      .1       0    4921     .05       0  7761.1      .1       0
  8181.1    .035       0  8197.2      .1       0  8355.7     .12       0
  8381.6      .1       0  9311.8     .08       0  9410.7      .1       0
Bank Sta=8181.1,8197.2
XS Rating Curve= 0 ,0
Exp/Cntr=0.3,0.1

Type RM Length L Ch R = 1 ,162150  ,890,890,890
BEGIN DESCRIPTION:
Black Creek 160.0
END DESCRIPTION:
XS GIS Cut Line= 4
       1974971.3     13609258.07      1973877.57     13606966.44
      1970218.71     13606211.23      1968527.96     13606263.25
#Sta/Elev= 30
  2239.4  717.07  2318.3  716.35  2528.8  715.36  2636.1  715.45  3452.5  715.22
  3556.3  714.54  4377.1  711.37  4844.7  711.26  4975.3  713.08  4995.7  710.81
  5069.3  710.65  5071.1  709.85  5085.4  710.65  5179.5  712.08  5848.8  713.37
    6221  712.89  6282.3  711.77  6939.3  717.46  7262.5  718.98  7395.2  718.99
  7561.2     717  7885.4  712.38  8019.2  712.46  8160.4  712.84  8181.5  711.76
  9150.3  719.82  9228.7   721.3  9248.8  720.51 10102.3  726.49 10206.2  725.87
#Mann= 14 ,-1 , 0
  2239.4      .1       0  2318.3     .05       0  2528.8      .1       0
  2636.1     .05       0  3452.5      .1       0  3556.3     .05       0
  4844.7      .1       0  5069.3     .07       0  5085.4      .1       0
  7561.2      .1       0  8019.2     .12       0  8160.4      .1       0
  9150.3     .08       0  9248.8      .1       0
Bank Sta=5069.3,5085.4
XS Rating Curve= 0 ,0
Exp/Cntr=0.3,0.1

Type RM Length L Ch R = 1 ,161260  ,1574,1574,1574
BEGIN DESCRIPTION:
Black Creek 162.0
END DESCRIPTION:
XS GIS Cut Line= 3
      1976853.27     13605982.06       1975214.8     13606123.12
      1968738.51     13606036.34
#Sta/Elev= 30
  1731.8  738.69  1950.9  732.68  2131.5  729.34  2322.2  721.75  2723.7  714.35
  2834.1  711.02  3506.1  706.78  3648.1  705.04  3649.9  704.24  3662.5  704.24
  3664.3  705.04  4769.1  709.63  4876.3  709.71  4896.3  710.62  4966.3  709.95
  4986.3  708.71  5016.2  710.07  5504.7  710.76  5716.3  710.88  5876.4  713.09
  6016.4  716.57  6606.4  716.73  7397.7  712.74  7656.5  711.14  7776.5  712.36
  7996.5   711.9  9002.5  720.09  9086.6  721.37  9107.3   720.8  9853.2  724.91
#Mann= 10 ,-1 , 0
  1731.8      .1       0  3648.1     .07       0  3664.3      .1       0
  4769.1      .1       0  5016.2     .05       0  5504.7      .1       0
  6016.4     .05       0  7397.7      .1       0  9002.5     .05       0
  9107.3      .1       0
Bank Sta=3648.1,3664.3
XS Rating Curve= 0 ,0
Exp/Cntr=0.3,0.1

Type RM Length L Ch R = 1 ,159686  ,1504,1504,1504
BEGIN DESCRIPTION:
Black Creek 163.0
END DESCRIPTION:
XS GIS Cut Line= 3
      1976831.57     13605678.24      1975529.47     13605743.35
      1968834.61     13605732.49
#Sta/Elev= 30
  3007.6  743.75  3184.4  739.87  3646.8  721.45  3955.4  711.97  4095.5  709.02
  4565.8  705.16  4791.5  705.77  4965.8  705.71    5007  702.25  5009.3  701.45
  5024.6  702.25  5025.8  704.12  5035.8  705.62  5224.3  707.01  5615.2  708.34
  5657.5  708.38  6625.8  708.81  7275.8  717.44  7585.8  715.22  7945.8  715.08
  8225.8  711.33  8265.8   712.5  8295.8  710.64  8385.8  709.45  8865.8  709.65
  9555.8  712.98 10340.1  722.59 10365.8  723.94 10416.9  722.71 11006.2  725.76
#Mann= 9 ,-1 , 0
  3007.6      .1       0  4791.5     .05       0    5007     .04       0
  5024.6     .05       0  5224.3      .1       0  5615.2     .05       0
  5657.5      .1       0 10340.1     .05       0 10416.9      .1       0
Bank Sta=5007,5024.6
XS Rating Curve= 0 ,0
Exp/Cntr=0.3,0.1

Type RM Length L Ch R = 1 ,158182  ,1832,1832,1832
BEGIN DESCRIPTION:
Black Creek 159.0
END DESCRIPTION:
XS GIS Cut Line= 3
      1977041.62     13605039.35      1972796.84     13604687.79
      1969529.26     13604232.15
#Sta/Elev= 30
  3317.5  725.83  4096.8  715.82  4207.2  713.41  4247.3  709.76  4275.6  712.41
  4367.7  711.36  4668.7  714.14  4864.4  706.45    4991  697.53  4993.4  696.73
  5008.7  697.53  5010.4   701.5  5049.2  701.58  5295.9  701.56    5730  704.52
  6700.4  704.47  6856.2  704.53  6896.3  701.96  6916.4  704.59  7606.6  709.68
  7717.8  708.83  8201.2  704.87  8777.9  706.34  9299.4  707.65  9662.1  718.43
  9876.8  718.72   10113  722.96 10415.9  724.95 10857.2  733.23   10876  734.13
#Mann= 12 ,-1 , 0
  3317.5      .1       0  4864.4     .16       0    4991     .07       0
  5008.7     .16       0  5049.2      .1       0  5295.9     .05       0
  6700.4      .1       0  7606.6     .05       0  7717.8      .1       0
  8201.2     .16       0  8777.9      .1       0 10857.2     .05       0
Bank Sta=4991,5008.7
XS Rating Curve= 0 ,0
Exp/Cntr=0.3,0.1

Type RM Length L Ch R = 1 ,156350  ,1879,1879,1879
BEGIN DESCRIPTION:
Black Creek 158.0
END DESCRIPTION:
XS GIS Cut Line= 3
      1976729.17     13603229.46      1973219.27     13603327.08
      1969854.11      13603008.1
#Sta/Elev= 30
  3453.1  730.18  3697.4  730.73  4377.6  709.81  4567.7  709.62  4627.7   705.2
  4647.7  709.12  4727.8  708.71  4845.4  700.71  5003.5  694.65  5209.3  697.65
  6346.7  701.75  6750.7  699.68  6858.6  699.77  6918.6  692.93    6964  698.94
    7049  700.91  7059.1  697.15  7060.1  692.21  7062.6  691.41  7078.1  692.21
  7089.2  697.79  7119.3  699.24  8207.1  701.47  8816.9  719.15  9449.7   713.1
  9489.9  708.75  9550.2  718.51  9590.3  713.59  9640.6  713.29 10344.6  722.92
#Mann= 7 ,-1 , 0
  3453.1      .1       0  4845.4     .16       0  5003.5      .1       0
  5209.3     .05       0  6750.7      .1       0  7060.1     .07       0
  7078.1      .1       0
Bank Sta=7060.1,7078.1
XS Rating Curve= 0 ,0
Exp/Cntr=0.3,0.1

Type RM Length L Ch R = 1 ,154471  ,1566,1566,1566
BEGIN DESCRIPTION:
Black Creek 157.0
END DESCRIPTION:
XS GIS Cut Line= 3
       1977906.3     13601726.53      1975036.42     13601719.04
      1970089.27     13601419.61
#Sta/Elev= 30
    1864  715.37  2615.3  701.91  3025.3  697.37  3625.3   694.1  4206.7  695.73
  4377.4  696.52  4605.3  696.49    4884  691.45  4925.6  691.25  4969.8  691.68
  4985.8  688.65  4986.8  684.49  4989.3  683.69  5004.8  684.49  5005.8  690.54
  5197.7   693.7  5466.7  697.31  6010.9  694.72  6109.3  690.82  6137.9   688.1
  6157.9  692.42  6207.6  692.34  6899.3  694.52  7109.7   701.9  7257.8  700.83
  7440.3   698.3  8171.6  702.97  8301.8  699.84  8502.2  705.78  9690.1  715.32
#Mann= 13 ,-1 , 0
    1864      .1       0  4206.7     .16       0  4377.4      .1       0
    4884     .16       0  4925.6      .1       0  4969.8     .16       0
  4986.8     .07       0  5004.8     .16       0  5197.7      .1       0
  6010.9     .05       0  6109.3     .16       0  6207.6     .05       0
  7257.8      .1       0
Bank Sta=4986.8,5004.8
XS Rating Curve= 0 ,0
Exp/Cntr=0.3,0.1

Type RM Length L Ch R = 1 ,152905  ,1643,1643,1643
BEGIN DESCRIPTION:
Black Creek 156.0
END DESCRIPTION:
XS GIS Cut Line= 2
      1977566.06      13600580.7      1970765.63     13599896.13
#Sta/Elev= 30
  2551.5  714.05  2743.5  714.71  3058.9  704.96  3286.3  702.39  3654.9  694.49
  3718.4  695.26  3755.1  692.77  3889.3  690.66  4572.7  693.17  4928.6  688.34
  4952.1  682.95  4974.7  686.01  4975.8  681.22  4978.3  680.42  4993.8  681.22
  5004.9     687  5048.1  687.28  5125.5  686.58  5406.9     690  5935.2  688.56
  6040.1  687.97  6080.3  681.95  6090.4  685.79  6110.5  684.66  6149.2  688.56
  6329.5   690.4    6428  690.15  7587.9     692  9144.3  713.57  9386.3  714.13
#Mann= 8 ,-1 , 0
  2551.5      .1       0  4928.6     .16       0  4975.8     .07       0
  4993.8     .16       0  5048.1      .1       0  5935.2     .12       0
  6329.5     .05       0    6428      .1       0
Bank Sta=4975.8,4993.8
XS Rating Curve= 0 ,0
Exp/Cntr=0.3,0.1

Type RM Length L Ch R = 1 ,151262  ,97,97,97
BEGIN DESCRIPTION:
Black Creek 155.0
END DESCRIPTION:
XS GIS Cut Line= 3
      1976956.78     13598977.07      1974652.22      13598811.4
      1971288.24     13598802.38
#Sta/Elev= 30
  2683.3   697.4  2923.3  694.83  3039.8  693.94  3138.2  692.85  3497.2  689.08
  4472.6  686.31  4614.4  685.68  4729.9   684.6  4734.9  685.59  4869.8  684.46
  4874.8   685.6  4940.9  685.03  4960.9  684.22    4971  678.94  5001.3  677.88
  5003.8  677.08  5020.7  677.88    5021  681.07    5031  683.25    5051  683.93
    5181   683.4  5718.4  686.99  5795.1  687.48  5893.4  687.31    6351  689.61
    6651  687.28    7011   688.7    7511  698.12    7841  701.63  8357.8  712.05
#Mann= 11 ,-1 , 0
  2683.3     .05       0  2923.3     .08       0  3039.8     .05       0
  3138.2      .1       0  4472.6     .05       0  4614.4     .08       0
  5001.3     .07       0  5020.7     .08       0  5718.4      .1       0
  5795.1     .05       0  5893.4      .1       0
Bank Sta=5001.3,5020.7
XS Rating Curve= 0 ,0
Exp/Cntr=0.3,0.1

Type RM Length L Ch R = 1 ,151165  ,1309,1309,1309
BEGIN DESCRIPTION:
Mapping XS 42406c9d
END DESCRIPTION:
XS GIS Cut Line= 3
      1977137.38     13598754.85       1974109.6     13598706.24
      1971310.96     13598609.01
#Sta/Elev= 30
  2503.1  706.74  2845.5  696.96  3135.6  691.79  3345.6  691.69  3575.6  688.34
  3605.6  689.38  3645.6   687.6  4017.3  686.81  4055.8  686.66  4065.7  687.88
  4195.7  686.11  4901.4  684.41  4945.8  683.33  4996.1   677.3  4998.6   676.5
  5015.5   677.3  5085.8  682.59  5485.9  685.72  5906.1  686.79  6166.2  689.54
  6616.5  686.33  6676.6  687.54  6867.3  686.75  6946.7  688.55  6996.8  687.87
  7016.8  689.45  7316.9  690.83    7387  693.38  7787.2  700.59  8331.6  714.04
#Mann= 5 ,-1 , 0
  2503.1      .1       0  4017.3     .05       0  4901.4      .1       0
  4996.1     .07       0  5015.5      .1       0
Bank Sta=4996.1,5015.5
XS Rating Curve= 0 ,0
Exp/Cntr=0.3,0.1

Type RM Length L Ch R = 1 ,149856  ,760,760,760
BEGIN DESCRIPTION:
Black Creek 154.0
END DESCRIPTION:
XS GIS Cut Line= 3
      1977317.94     13597921.51      1974081.82     13597588.18
      1971781.22     13597604.46
#Sta/Elev= 30
  2670.6  737.56  3266.3   707.7  3563.5  696.05  3960.3  685.71    4372  684.18
  4573.6  682.84  4633.1  683.62  4869.1  680.21  4933.6  679.72  4975.7  679.22
  4985.7  675.72  4986.1  674.59  4988.6  673.79  5005.5  674.59  5005.8  678.87
  5032.2  679.91  5056.1  678.45  5216.9  682.43  5528.6  683.58  5548.7   682.6
  5811.8  682.32  6504.8  683.03  6634.4  683.46  7154.7  686.04  7280.7  685.78
  7300.7   687.6  7410.7  690.42  7440.7  689.67  7590.1  692.67  8224.5  699.33
#Mann= 10 ,-1 , 0
  2670.6      .1       0    4372     .05       0  4869.1      .1       0
  4933.6     .07       0  4986.1     .07       0  5005.5     .07       0
  5032.2     .05       0  6504.8      .1       0  6634.4     .05       0
  7154.7      .1       0
Bank Sta=4986.1,5005.5
XS Rating Curve= 0 ,0
Exp/Cntr=0.3,0.1

Type RM Length L Ch R = 1 ,149096  ,1629,1629,1629
BEGIN DESCRIPTION:
Black Creek 153.0
END DESCRIPTION:
XS GIS Cut Line= 3
      1977060.98     13597011.79      1975394.32     13597004.85
      1971970.72     13597018.74
#Sta/Elev= 30
  3059.8  708.48  3845.8  692.33  4075.8  688.89  4185.8  688.76  4215.8   686.8
  4495.8  684.61  4555.8  683.24  4715.8   682.8  4885.8  678.98  4905.8  679.82
  4925.8  678.11  4975.8  678.02    4986  672.71  4988.5  671.91  5005.5  672.71
  5005.8  677.49  5015.8   679.5  5106.3  678.15  5405.8  681.15  6035.8  679.64
  6785.8  681.34  7015.8  684.54  7291.7  685.54  7365.8  686.15  7395.8  688.95
  7465.8  690.62  7535.8  693.83  7605.8  691.99  7725.8  693.56  8150.1  695.81
#Mann= 5 ,-1 , 0
  3059.8      .1       0    4986     .07       0  5005.5      .1       0
  5106.3     .05       0  7291.7      .1       0
Bank Sta=4986,5005.5
XS Rating Curve= 0 ,0
Exp/Cntr=0.3,0.1

Type RM Length L Ch R = 1 ,147467  ,1803,1803,1803
BEGIN DESCRIPTION:
Mapping XS 1339d556
END DESCRIPTION:
XS GIS Cut Line= 4
      1976097.44     13595933.67      1974795.36     13595816.48
      1973610.46     13596545.65      1971749.23     13596558.66
#Sta/Elev= 30
  3378.2  700.02  3561.4  697.99  4003.2  689.12  4193.9   683.6  4254.2  680.06
  4887.3  677.87  4976.1   674.5  4981.9  673.28  4987.6  668.53  4990.1  667.73
  5007.1  668.53  5012.7  675.45  5018.6  675.95    5034  674.87  5085.2   675.7
  5128.7  678.31  5390.5  677.17  5470.7  675.07  5727.2  677.87  6342.3  679.62
  6682.3  683.29  6762.3  685.43  6875.7  684.25  6892.3  683.75  6912.3  685.72
  7072.3  689.08  7162.3  689.35  7202.3  690.87  7402.3  690.28  7938.1  692.99
#Mann= 5 ,-1 , 0
  3378.2      .1       0  4987.6     .07       0  5007.1      .1       0
  5727.2     .05       0  6875.7      .1       0
Bank Sta=4987.6,5007.1
XS Rating Curve= 0 ,0
Exp/Cntr=0.3,0.1

Type RM Length L Ch R = 1 ,145664  ,1007,1007,1007
BEGIN DESCRIPTION:
Black Creek 152.0
END DESCRIPTION:
XS GIS Cut Line= 3
      1976891.67      13595582.1       1974196.4     13595126.38
        1971525.       13595525.
#Sta/Elev= 30
  1401.4  705.85  1864.6   702.5  2133.5  697.77    2686  682.68  3048.9  679.66
  3090.1  678.27  3385.8  676.76  4652.1  673.71  4767.7  672.89  4867.7  671.67
  4965.4   672.6  4971.5  670.41  4976.6  671.18  4985.6  668.32  4985.9  664.83
  4988.4  664.03  5005.7  664.83  5005.9  670.12    5016  673.11  5056.4  676.13
  5076.6  675.77    5105  679.44  5157.5   680.4  5243.5  677.49  5248.6  676.09
  5312.8  680.14  5875.4  684.87  6047.3  688.08  6542.7  693.28  6835.9  694.91
#Mann= 7 ,-1 , 0
  1401.4      .1       0  3048.9     .05       0  4652.1      .1       0
  4767.7     .16       0  4867.7      .1       0  4985.9     .07       0
  5005.7      .1       0
Bank Sta=4985.9,5005.7
XS Rating Curve= 0 ,0
Exp/Cntr=0.3,0.1

Type RM Length L Ch R = 1 ,144657  ,571,571,571
BEGIN DESCRIPTION:
Black Creek 151.0
END DESCRIPTION:
XS GIS Cut Line= 4
      1977126.13     13594905.03      1975290.15     13594683.67
        1973725.       13594425.      1971958.42     13594410.24
#Sta/Elev= 30
  1549.8  715.47  2004.2  709.11  2347.7  700.35  2593.9  691.97  2799.9  687.19
  3353.9  679.38  3414.4   679.8  3440.6  678.26  3779.3  674.39  4280.6  674.23
  4719.2  671.68  4818.4  671.28  4896.4  669.41  4914.5  665.67  4924.6  665.48
  4944.9  669.87  4975.3  670.13  4985.5  667.23  4985.6   664.7  4988.1   663.9
  5005.4   664.7  5007.5  666.19  5015.5  669.53  5175.5  677.11  5435.5  682.63
  5715.5  683.79  5835.5   681.7  5995.5  681.41  6475.5  687.17  6752.1  688.99
#Mann= 7 ,-1 , 0
  1549.8      .1       0  3440.6     .05       0  4719.2     .12       0
  4818.4     .16       0  4985.6     .07       0  5005.4     .16       0
  5007.5      .1       0
Bank Sta=4985.6,5005.4
XS Rating Curve= 0 ,0
Exp/Cntr=0.3,0.1

Type RM Length L Ch R = 1 ,144086  ,555,555,555
BEGIN DESCRIPTION:
Black Creek 150.0
END DESCRIPTION:
XS GIS Cut Line= 3
      1976657.34     13593433.67        1973875.       13593925.
      1971110.43     13593811.27
#Sta/Elev= 30
  2180.5  693.38  2396.1  690.17  3021.3  684.88    3178  682.78    3199   681.4
  3228.8  682.92  3381.1  682.28  3411.6  683.95  3442.1  688.53  3484.9  683.53
  3639.1  680.36  3838.1  674.82  4110.9  671.38  4759.4   671.3  4873.3   669.5
  4924.7  667.45  4965.3   668.1  4978.8  666.54  4985.8  662.76  4988.3  661.96
  5005.6  662.76  5005.9   665.9  5015.9  667.92    5086   668.4    5196  673.72
  5396.2  680.54  5617.8  677.81  6086.8  677.88    7518  687.96  7772.8  688.61
#Mann= 6 ,-1 , 0
  2180.5      .1       0  3639.1     .05       0  4759.4      .1       0
  4873.3     .16       0  4985.8     .07       0  5005.6      .1       0
Bank Sta=4985.8,5005.6
XS Rating Curve= 0 ,0
Exp/Cntr=0.3,0.1

Type RM Length L Ch R = 1 ,143531  ,1426,1426,1426
BEGIN DESCRIPTION:
Black Creek 149.0
END DESCRIPTION:
XS GIS Cut Line= 3
      1976024.97     13592625.01        1973825.       13593425.
      1971175.52     13593355.54
#Sta/Elev= 30
  2675.9  713.18  2739.7  712.54  2894.7  705.53  3005.7  702.58  3245.8  693.31
  3314.3  692.25  3652.8  679.46  3800.5  677.04    3831   675.2  3861.6  675.15
  4090.4  668.47  4502.7  670.19  4711.6  669.31  4899.8  666.05  4947.1  666.52
  4963.6  665.35  4970.9   662.9  4976.2  665.37  4984.9  664.18  4985.6  660.76
  4988.1  659.96  5002.9  659.96  5005.4  660.76  5014.2  666.26  5046.8  668.65
  5126.8  670.76  5356.9  674.11  5757.1  675.03  6167.2  677.93  7667.2  684.39
#Mann= 5 ,-1 , 0
  2675.9      .1       0  4947.1     .16       0  4984.9      .1       0
  4985.6     .07       0  5005.4      .1       0
Bank Sta=4985.6,5005.4
XS Rating Curve= 0 ,0
Exp/Cntr=0.3,0.1

Type RM Length L Ch R = 1 ,142105  ,237,237,237
BEGIN DESCRIPTION:
Black Creek 148.0
END DESCRIPTION:
XS GIS Cut Line= 5
      1976040.17     13592524.81      1974831.82      13592476.2
      1974435.99     13592260.92      1973584.42     13592405.02
      1971370.89     13592873.77
#Sta/Elev= 30
  3459.4  710.19  3554.6  709.75  3624.7  705.74  3654.7  707.45  3724.8  707.01
  4335.3  679.98  4475.4  676.49  4655.5  669.88  4843.9  665.44  4926.9  663.01
  4954.6  664.92  4976.4  664.22  4982.6  659.73  4985.1  658.93  5002.6  659.73
  5006.6  664.41  5083.3   665.2    5313  668.23  5708.3  667.11  6268.6  672.16
  6309.5  670.63  6345.1  672.46  6350.4  671.43  6638.1  672.93  6677.5   674.6
  6943.2  678.64  7169.4  680.41  7525.9  680.54  7924.5  690.49  8245.6   690.4
#Mann= 5 ,-1 , 0
  3459.4      .1       0  4843.9     .16       0  4982.6     .07       0
  5002.6     .16       0  5083.3      .1       0
Bank Sta=4982.6,5002.6
XS Rating Curve= 0 ,0
Exp/Cntr=0.3,0.1

Type RM Length L Ch R = 1 ,141868  ,1233,1233,1233
BEGIN DESCRIPTION:
Mapping XS d492dd05
END DESCRIPTION:
XS GIS Cut Line= 5
      1976054.01     13592441.47      1974887.37     13592240.09
      1974491.54     13592045.65      1973692.93     13592184.53
      1971199.96     13592448.41
#Sta/Elev= 30
  3597.1  707.36  3880.2   705.1    4002  701.81  4377.5  682.76  4779.7  671.09
  4895.7  665.75    4937  663.11  4942.6  664.16  4959.5  662.64    4973  663.42
    4982  662.41  4985.3  660.63  4987.8  659.83  5005.3  660.63  5017.6  664.16
  5026.9  664.59  5115.2   663.8    5391  667.64  5837.6  666.96  5878.2  664.21
  5908.7  666.94  6010.7  668.45  6724.4  671.08  6965.7  675.54  7223.3  682.41
  7413.9  684.91  7870.7  682.66  7991.4   684.8  8222.7   685.1  8539.5  689.54
#Mann= 5 ,-1 , 0
  3597.1      .1       0  4895.7     .16       0  4985.3     .07       0
  5005.3     .16       0  5115.2      .1       0
Bank Sta=4985.3,5005.3
XS Rating Curve= 0 ,0
Exp/Cntr=0.3,0.1

Type RM Length L Ch R = 1 ,140635  ,1147,1147,1147
BEGIN DESCRIPTION:
Black Creek 147.0
END DESCRIPTION:
XS GIS Cut Line= 3
      1975811.84     13591181.06      1974657.34     13591085.58
      1970984.96     13591868.72
#Sta/Elev= 30
  3966.8  686.84  4053.9  686.03  4184.4   680.3  4284.7  678.99    4375  675.18
  4686.1  668.22  4859.4  667.37  4916.9  665.18  4946.1  662.34  4977.1  662.29
  4987.1   661.3  4987.2  659.24  4989.7  658.44  5007.2  659.24  5027.3   662.9
  5129.4  661.35  5158.3  663.02  5270.8  661.41  5436.8  665.05  6410.8  665.67
  6772.7  665.77  7314.7  670.35  7396.2  671.02  7428.2  672.94  7520.3  672.22
  7990.6  676.12  8491.6     688  8598.8  688.76  8808.6  686.99  8880.2  688.37
#Mann= 7 ,-1 , 0
  3966.8      .1       0  4859.4     .16       0  4987.2     .07       0
  5007.2     .16       0  5129.4      .1       0  6410.8     .05       0
  7314.7      .1       0
Bank Sta=4987.2,5007.2
XS Rating Curve= 0 ,0
Exp/Cntr=0.3,0.1

Type RM Length L Ch R = 1 ,139488  ,657,657,657
BEGIN DESCRIPTION:
Black Creek 146.0
END DESCRIPTION:
XS GIS Cut Line= 3
      1975953.35     13590206.24        1974225.       13590275.
       1971710.4     13590940.12
#Sta/Elev= 30
  3234.5  691.63  3320.4  692.78  3356.6  693.73  3474.9  694.78  3523.1  692.56
  3692.9  676.38  3830.3     674  3913.4  675.84    4337  676.98  4587.9  674.56
  4728.6  668.88  4884.2  659.67  4924.2  660.32  4934.2  659.14  4971.4  660.78
  4974.6  660.78  4976.8  653.83  4979.3  653.03    4997  653.83  5005.6  657.16
  5027.2  660.56  5097.3  659.77  5119.4  657.81  5142.7  659.92  5233.2  661.21
    5835  663.07  6152.8  661.83  6746.1  665.51    7133  671.69  7565.3   675.2
#Mann= 11 ,-1 , 0
  3234.5      .1       0  3320.4     .16       0  3356.6      .1       0
  3474.9     .16       0  3692.9      .1       0  4728.6     .07       0
  4971.4      .1       0  4976.8     .07       0    4997      .1       0
    5835     .05       0  6746.1      .1       0
Bank Sta=4976.8,4997
XS Rating Curve= 0 ,0
Exp/Cntr=0.3,0.1

Type RM Length L Ch R = 1 ,138831  ,901,901,901
BEGIN DESCRIPTION:
Black Creek 145.0
END DESCRIPTION:
XS GIS Cut Line= 3
      1974974.98       13589875.      1973475.92     13589870.73
      1971722.46     13590365.52
#Sta/Elev= 30
  3812.9  676.45  3912.9  678.74  4052.9  678.02  4132.9   674.7  4222.9  668.58
  4292.9   666.2  4412.9  665.25  4562.9  662.01  4672.9  662.46  4741.6  659.95
  4934.3  658.51  4952.9  658.26  4962.9  654.99  4982.8  651.92  4985.3  651.12
    5003  651.92  5012.9  656.78  5022.9  658.19  5112.9  656.79  5132.9  658.05
    5396  660.76  5666.2   658.9    5874  660.79  6258.5  667.33  6403.9  667.55
  6450.7  665.24  6529.1  664.12  6642.9  664.32  6861.1  665.83  7133.9   669.7
#Mann= 5 ,-1 , 0
  3812.9      .1       0  4741.6     .12       0  4934.3      .1       0
  4982.8     .07       0    5003      .1       0
Bank Sta=4982.8,5003
XS Rating Curve= 0 ,0
Exp/Cntr=0.3,0.1

Type RM Length L Ch R = 1 ,137930  ,659,659,659
BEGIN DESCRIPTION:
Black Creek 144.0
END DESCRIPTION:
XS GIS Cut Line= 4
      1975810.96     13589697.11      1974283.21     13589254.41
      1972911.68      13589124.2      1971435.95     13589566.92
#Sta/Elev= 30
  2496.5  673.28  3616.7  668.34  4012.4  663.71  4063.1  661.89  4296.2  662.84
  4477.1  658.46  4718.1  659.89  4800.4  658.61  4897.1  657.68  4982.3  655.85
  4989.3  655.08  4999.3  649.74  5001.8  648.94  5019.6  649.74  5029.5  655.61
  5039.6  656.01  5069.7   654.7  5119.9   657.2  5220.4  655.76  5320.8  657.34
  5399.8  661.01  5464.8  661.95  5552.3  667.27  5711.9  670.75  5942.1  670.79
  5962.5  672.09    6003  670.17  6321.4  665.72  6933.4  670.29  7005.5  669.62
#Mann= 5 ,-1 , 0
  2496.5      .1       0  4800.4     .12       0  4897.1      .1       0
  4999.3     .07       0  5019.6      .1       0
Bank Sta=4999.3,5019.6
XS Rating Curve= 0 ,0
Exp/Cntr=0.3,0.1

Type RM Length L Ch R = 1 ,137271  ,115,115,115
BEGIN DESCRIPTION:
Black Creek 143.0
END DESCRIPTION:
XS GIS Cut Line= 4
      1976171.24     13589098.17      1974048.83     13588551.29
      1972764.11     13588607.71      1971692.09     13589245.72
#Sta/Elev= 30
  1939.4  678.51  2100.7  677.44  2431.2  670.45  2571.9  666.34  2947.5  660.22
    3172  659.32  3463.9  659.73  3567.1  661.88  3639.4  661.85    3753  659.04
  3866.6  658.89  4056.9  661.19  4265.1  656.66  4794.5  657.27  4855.7  656.69
  4895.7  654.31  4965.8  653.03  4985.6  649.44  4988.1  648.64  5003.4  648.64
  5005.9  649.44  5012.1  654.52  5045.8  653.56  5276.1     661  5823.3  670.35
  6033.2  670.92    6347  665.96  6420.7   666.7  6500.6  665.96  6664.6  667.89
#Mann= 4 ,-1 , 0
  1939.4      .1       0  4794.5     .07       0  4985.6     .07       0
  5005.9      .1       0
Bank Sta=4985.6,5005.9
XS Rating Curve= 0 ,0
Exp/Cntr=0.3,0.1

Type RM Length L Ch R = 1 ,137156  ,824,824,824
BEGIN DESCRIPTION:
Black Creek 142.0
END DESCRIPTION:
XS GIS Cut Line= 5
      1976480.22     13588888.95      1974556.89     13588319.58
      1973142.58     13588489.66      1972817.06     13588363.79
      1971551.43     13589157.19
#Sta/Elev= 30
  1628.3  682.28  2051.7  671.17    2295  668.26  2361.5  668.99  2438.4  666.77
  2996.6  658.82  3187.7  657.65  3867.7  658.93  4290.7   655.5  4774.2  658.01
  4965.6  654.08  4974.2  653.67  4985.6  649.26  4988.1  648.46  5005.9  649.26
    5026  652.28  5058.6  651.27  5084.1  653.31  5089.5  651.84  5108.7  654.46
  5270.5  659.41  5313.4  660.22  5337.6  657.98  5445.5  662.97  5490.7  661.62
  5527.3  663.96  5904.4     669  6512.5  667.39  6591.4  665.79  6901.4  667.93
#Mann= 3 ,-1 , 0
  1628.3      .1       0  4985.6     .07       0  5005.9      .1       0
Bank Sta=4985.6,5005.9
XS Rating Curve= 0 ,0
Exp/Cntr=0.3,0.1

Type RM Length L Ch R = 1 ,136332  ,845,845,845
BEGIN DESCRIPTION:
Black Creek 141.0
END DESCRIPTION:
XS GIS Cut Line= 4
      1976275.02       13587875.      1975173.83     13587582.54
      1972647.79       13587869.      1971762.35     13588494.01
#Sta/Elev= 30
  1867.5  701.58  2022.7  696.36  2120.9  690.97  2311.4  674.47  2488.3  661.72
  2592.6  656.54  2702.8  653.03  2850.5  651.36  2881.5  652.17  3072.1  651.42
  3508.9  654.92    4002  653.33  4132.9  653.61  4344.2  655.88  4595.8  655.31
  4706.5  657.03  4861.2  654.79  4948.1   653.5  4978.2  650.16  4988.2  646.21
  4990.7  645.41  5008.5  646.21  5018.5  652.73  5046.3  653.23  5129.2  653.23
  5441.2  662.29  5613.7  664.62  5777.6  664.85    6238   662.5  6632.9  663.88
#Mann= 5 ,-1 , 0
  1867.5      .1       0  4861.2     .12       0  4988.2     .07       0
  5008.5     .12       0  5046.3      .1       0
Bank Sta=4988.2,5008.5
XS Rating Curve= 0 ,0
Exp/Cntr=0.3,0.1

Type RM Length L Ch R = 1 ,135487  ,1404,1404,1404
BEGIN DESCRIPTION:
Mapping XS b993c6b8
END DESCRIPTION:
XS GIS Cut Line= 4
      1975962.65     13586961.89      1973914.03     13586901.13
      1972646.67     13587126.82      1971822.28     13588350.39
#Sta/Elev= 30
  2177.4  687.69  2445.2   680.4  2535.2  676.31  2825.3   657.6  2955.4  652.09
  3035.4  650.58  3256.8  650.35  3485.6  653.04  3655.7  651.41  4005.9  651.99
  4025.9  653.62  4055.9  651.98    4744  654.93  4865.9  651.84  4962.2  652.48
  4977.6  650.51  4987.7  645.07  4990.2  644.27    5008  645.07  5021.1  649.35
  5038.5  651.85  5048.7   650.7  5075.1  650.92  5231.5     654  5585.1  652.43
  5765.2   655.9    5810  655.56    5846  657.31  6025.9  658.98  6989.6  662.95
#Mann= 3 ,-1 , 0
  2177.4      .1       0  4987.7     .07       0    5008      .1       0
Bank Sta=4987.7,5008
XS Rating Curve= 0 ,0
Exp/Cntr=0.3,0.1

Type RM Length L Ch R = 1 ,134083  ,1251,1251,1251
BEGIN DESCRIPTION:
Black Creek 140.0
END DESCRIPTION:
XS GIS Cut Line= 3
      1975745.62     13586284.81      1973028.61     13585790.02
      1970511.25     13583915.01
#Sta/Elev= 30
    2393  671.66  2759.7  661.04  3028.5   658.5  3148.2  655.62  3254.8  651.58
  3389.7  649.36  4812.8  651.83  4849.1  650.19  4894.1  648.47  4914.4  649.93
  4935.7  647.06  4944.9  647.07  4965.2  649.83  4975.4  649.31  4983.9  647.46
  4985.6  644.56  4988.1  643.76  5005.9  644.56  5016.1  649.04  5024.9  651.07
  5087.2  652.14  5383.2  648.88  5639.7  648.07  5904.6  651.63  6671.1  655.27
  6876.4  655.93  7126.6  658.81  7935.7  674.67  8253.6  676.33  8293.6     677
#Mann= 9 ,-1 , 0
    2393      .1       0  3028.5     .05       0  4849.1      .1       0
  4985.6     .07       0  5005.9      .1       0  5024.9     .05       0
  6671.1      .1       0  7935.7     .05       0  8253.6      .1       0
Bank Sta=4985.6,5005.9
XS Rating Curve= 0 ,0
Exp/Cntr=0.3,0.1

Type RM Length L Ch R = 1 ,132832  ,254,254,254
BEGIN DESCRIPTION:
Black Creek 139.0
END DESCRIPTION:
XS GIS Cut Line= 6
      1976101.04     13585148.26      1973905.35     13584487.93
      1973193.54     13584730.99      1972776.88     13584800.43
      1972221.32     13584540.02      1970798.86     13583941.54
#Sta/Elev= 30
  1678.5  692.46  1813.3  690.52  2329.6  671.98  2770.8  664.51  2948.3  659.72
    3742  656.08  3756.7  657.32  4071.3  648.23  4097.4  649.83  4102.6  652.45
  4109.1   653.3  4172.5  644.21  4360.6  647.88  4818.9  649.46  4914.6  649.26
  4975.5  644.77  4985.1  641.83  4987.7  641.03  5006.4  641.83    5016  646.89
  5036.3  646.39  5082.2  648.97  5189.6   651.5  5258.4  652.57  5417.6  651.62
  6243.7  654.85  6820.4  663.53  6973.7   668.5  7256.1  672.25  7302.7   673.3
#Mann= 8 ,-1 , 0
  1678.5      .1       0  4360.6     .05       0  4818.9      .1       0
  4985.1     .07       0  5006.4      .1       0  5189.6     .05       0
  5417.6      .1       0  7256.1     .05       0
Bank Sta=4985.1,5006.4
XS Rating Curve= 0 ,0
Exp/Cntr=0.3,0.1

Type RM Length L Ch R = 1 ,132578  ,468,468,468
BEGIN DESCRIPTION:
Black Creek 138.0
END DESCRIPTION:
XS GIS Cut Line= 6
      1975401.05     13584848.27      1973887.99     13584340.37
      1973228.27     13584540.02      1972672.71     13584531.34
      1972098.72     13583719.03      1970929.01     13583810.77
#Sta/Elev= 30
  2437.2  670.37  2655.8   667.6  2992.1   660.4  3287.4  658.48  3438.9     660
  3793.8  657.55  4206.7  647.21  4255.8  646.87  4277.8  650.76  4318.4  644.43
  4328.9  644.23  4349.8  644.41  4381.8  650.41  4409.5  646.91  4835.8  648.91
  4945.8  645.61  4965.8  646.69  4975.1  641.24  4977.7  640.44  4996.4  641.24
  5015.8     647  5055.8  649.09  5295.1  651.04  5924.3  651.64  6166.3  652.66
  6284.6   656.4  6350.2   656.4  6611.2  656.11    6804  658.05  7459.8  670.34
#Mann= 7 ,-1 , 0
  2437.2      .1       0  4975.1     .07       0  4996.4      .1       0
  5924.3     .05       0  6284.6      .1       0  6350.2     .05       0
    6804      .1       0
Bank Sta=4975.1,4996.4
XS Rating Curve= 0 ,0
Exp/Cntr=0.3,0.1
