HEC-RAS study Black Creek.prj: Black Creek Base Level Engineering

--- Black Creek.g01 (geometry) --- (continued)

Type RM Length L Ch R = 1 ,132110  ,354,354,354
BEGIN DESCRIPTION:
Mapping XS 11a5a352
END DESCRIPTION:
XS GIS Cut Line= 6
      1974263.58     13583800.03      1973300.04     13584018.78
      1972919.83     13584430.24      1972643.79      13584341.7
        1972149.     13583695.86      1971108.69     13583711.47
#Sta/Elev= 30
    3799  659.81  4314.8  647.86  4740.3  647.32  4749.8  644.73  4809.6  641.84
  4859.8  646.34  4895.5  646.63  4923.8  645.98  4930.6  643.87    4938  644.71
  4948.1  639.97  4950.9  639.17  4969.8  639.97  4987.3  642.29  4994.7  640.85
  5001.5  643.78  5015.7  642.03  5022.5   644.7    5044  644.87  5050.8  647.31
  5058.2  646.29    5065  648.39  5249.3  647.22  5670.2  650.27  6081.5  650.15
  6305.7  651.95  6446.3  655.73  6547.3  657.01  6957.3  657.08  7513.7  666.54
#Mann= 5 ,-1 , 0
    3799      .1       0  4948.1     .07       0  4969.8      .1       0
  6081.5     .05       0  6446.3      .1       0
Bank Sta=4948.1,4969.8
XS Rating Curve= 0 ,0
Exp/Cntr=0.3,0.1

Type RM Length L Ch R = 1 ,131756  ,1006,1006,1006
BEGIN DESCRIPTION:
Mapping XS 8c0d44e4
END DESCRIPTION:
XS GIS Cut Line= 6
      1974180.23      13583654.2      1973471.91     13583737.53
      1972862.54     13584331.28      1972701.08     13584310.45
      1972180.25     13583602.11      1971139.31     13583633.34
#Sta/Elev= 30
  4059.2  657.88  4280.5  653.57  4450.8  648.54  4506.2  647.64  4605.6  647.53
  4638.2  647.39  4781.9  647.32    4805  648.27  4882.2  646.59  4932.4  643.75
    4947  645.21  4961.7  643.87  4967.9  647.31  4976.3  644.98  4980.2  640.05
  4982.9  639.25  5001.9  640.05  5004.2  642.63  5018.1  645.07  5032.7  643.95
  5082.9  647.18  5460.4  647.04  5788.4  649.54  6194.8  649.23  6408.2  651.15
  6422.9  652.56  6535.4  654.54  6757.4  658.44  7217.6  657.64  7713.5  666.19
#Mann= 9 ,-1 , 0
  4059.2      .1       0  4450.8     .05       0  4506.2      .1       0
  4605.6     .05       0  4638.2      .1       0  4980.2     .07       0
  5001.9      .1       0  6194.8     .05       0  6535.4      .1       0
Bank Sta=4980.2,5001.9
XS Rating Curve= 0 ,0
Exp/Cntr=0.3,0.1

Type RM Length L Ch R = 1 ,130750  ,1041,1041,1041
BEGIN DESCRIPTION:
Black Creek 136.0
END DESCRIPTION:
XS GIS Cut Line= 4
      1974410.53     13583892.41      1973691.81     13583038.28
      1972572.02     13583038.28      1971718.97     13583267.15
#Sta/Elev= 30
  3152.7  662.84    3247  660.72  3396.6  659.71  3438.2  657.39    3446  658.46
  3474.6   658.3  3612.2   655.8    3729  654.21  3739.6  654.12    4103  647.64
  4126.1  647.27  4205.5  646.19  4400.2  646.24  4733.7  645.35  4755.4  644.89
    4892  643.11  4925.8  641.82  4945.8  644.48  4975.8  645.01  4984.9   637.9
  4987.7   637.1  5006.6   637.9  5015.8  642.24  5025.8  644.54  5215.8  643.69
  5325.8  644.39    5628  651.07  5817.6   657.4  6058.7  662.87    6272  660.91
#Mann= 12 ,-1 , 0
  3152.7      .1       0  3612.2     .05       0    3729      .1       0
  3739.6     .05       0    4103      .1       0  4126.1     .05       0
  4400.2      .1       0  4733.7     .05       0  4755.4      .1       0
    4892     .12       0  4984.9     .07       0  5006.6      .1       0
Bank Sta=4984.9,5006.6
XS Rating Curve= 0 ,0
Exp/Cntr=0.3,0.1

Type RM Length L Ch R = 1 ,129709  ,541,541,541
BEGIN DESCRIPTION:
Black Creek 135.0
END DESCRIPTION:
XS GIS Cut Line= 4
      1974509.49       13583882.      1973618.89     13582793.49
      1972743.89     13582116.41      1972608.47     13581283.04
#Sta/Elev= 30
    2669  664.07  2875.9  661.17  2911.1  661.86  2947.7     660  3104.9  658.44
  3409.2  654.42    3743   647.2  3889.2  645.95  3978.6  645.76  4376.4  645.29
  4704.1  641.97  4768.4  643.05  4917.8  641.82  4946.8  642.71  4975.8  642.05
  4990.3  640.08  4992.5   635.8  4995.3     635  5014.2   635.8  5017.4  640.22
  5025.6  643.38  5081.7  641.77    5175  643.63  5335.5  642.92  5365.6  641.29
  5375.7  642.67  5581.8  646.24  5841.8  654.78  5922.8  655.56  6026.1  658.39
#Mann= 7 ,-1 , 0
    2669      .1       0  3104.9     .05       0    3743      .1       0
  3889.2     .05       0  3978.6      .1       0  4992.5     .07       0
  5014.2      .1       0
Bank Sta=4992.5,5014.2
XS Rating Curve= 0 ,0
Exp/Cntr=0.3,0.1

Type RM Length L Ch R = 1 ,129168  ,633,633,633
BEGIN DESCRIPTION:
Black Creek 134.0
END DESCRIPTION:
XS GIS Cut Line= 4
      1974457.45     13583387.27      1974030.35     13582684.12
      1973308.88     13581991.12      1972785.57     13581095.59
#Sta/Elev= 30
  3166.2  659.53  3241.9  659.35    3542  655.53  3769.7  650.75  4048.7   645.4
  4734.6  645.36  4819.5  644.56  4920.6  641.93  4946.9  642.64  4953.8  642.04
    4961     640  4967.9  639.21  4977.7  636.07  4980.4  635.27  4996.6  635.27
  4999.4  636.07  5004.5  639.12  5008.8  640.33  5051.3  640.86  5063.2  640.31
  5167.6   641.7  5216.4  642.07  5319.4  640.74  5378.1  641.53  5661.6   649.6
  5677.4   649.2  5763.3  652.87  5794.7  653.35    5822  655.25  6026.5  660.65
#Mann= 9 ,-1 , 0
  3166.2      .1       0  3241.9     .05       0  3769.7      .1       0
  4920.6     .07       0  4977.7     .07       0  4999.4     .07       0
  5008.8     .16       0  5051.3     .12       0  5167.6      .1       0
Bank Sta=4977.7,4999.4
XS Rating Curve= 0 ,0
Exp/Cntr=0.3,0.1

Type RM Length L Ch R = 1 ,128535  ,650,650,650
BEGIN DESCRIPTION:
Black Creek 133.0
END DESCRIPTION:
XS GIS Cut Line= 3
      1975014.71     13583241.38      1973827.23     13581699.74
      1972885.59     13580648.86
#Sta/Elev= 30
  2967.9  653.93  3200.9   652.2  3278.9  652.71  3432.9  650.84  3747.9  650.69
  4170.3  643.59  4912.3  643.53  4925.8  643.51  4960.9  639.85  4982.6  638.64
  4985.8  635.38  4988.7  634.58    5005  634.58  5007.8  635.38  5011.1  638.08
    5032  639.88  5238.8  640.07  5242.1  639.87  5420.1  641.18  5690.6   646.3
  5761.6  649.64  5839.4  649.88  5938.8   652.9  6059.2  654.86  6065.9  655.96
  6101.8  656.42  6129.4  658.76  6193.8  660.48  6214.7  662.24  6324.9  665.19
#Mann= 9 ,-1 , 0
  2967.9      .1       0  3432.9     .05       0  3747.9      .1       0
  4912.3     .16       0  4985.8     .07       0  5007.8     .16       0
  5238.8      .1       0  5242.1     .16       0  5420.1      .1       0
Bank Sta=4985.8,5007.8
XS Rating Curve= 0 ,0
Exp/Cntr=0.3,0.1

Type RM Length L Ch R = 1 ,127885  ,669,669,669
BEGIN DESCRIPTION:
Black Creek 132.0
END DESCRIPTION:
XS GIS Cut Line= 3
      1975405.37     13583033.11       1974061.6     13581038.28
      1973651.29     13580508.51
#Sta/Elev= 30
  2807.3  654.31  3239.1  648.85  4037.5  642.24  4499.2   641.9  4878.8  638.73
  4975.3  639.85  4988.1  638.76    4992  633.21  4994.9  632.41    5014  633.21
    5018  638.14  5047.7   638.1  5109.8  643.33  5161.9  645.12  5211.5  649.83
  5241.7  650.81    5248  649.23  5268.9  649.82  5312.3  655.08  5569.5  663.17
  5611.1  662.87  5640.1  666.97  5675.4  666.98  5747.8  670.06  5783.1  670.35
  5789.4  668.74  5797.6  669.97  5803.9  668.09  5824.8  671.84  5882.6  672.63
#Mann= 5 ,-1 , 0
  2807.3      .1       0  4878.8     .16       0    4992     .07       0
    5014     .16       0  5109.8      .1       0
Bank Sta=4992,5014
XS Rating Curve= 0 ,0
Exp/Cntr=0.3,0.1

Type RM Length L Ch R = 1 ,127216  ,2399,2399,2399
BEGIN DESCRIPTION:
Black Creek 131.0
END DESCRIPTION:
XS GIS Cut Line= 3
      1976019.08     13583051.33      1975472.19     13581844.71
      1974057.27     13580160.69
#Sta/Elev= 30
  2564.8  660.83  3296.4  647.46  3428.1  646.03  3508.9  647.62  3834.4  641.28
  4072.1  640.83  4384.7  637.15  4682.6  639.67  4837.1  637.64  4966.2  638.05
  4980.5  637.06    4987  634.97  4990.3  631.39  4993.2  630.59  5012.3  631.39
  5015.6  635.28  5023.4  637.45  5029.9  636.07  5235.5  641.19  5257.5  644.01
  5327.8   645.5  5448.8  653.38  5604.9  658.17  5647.8   661.3  5725.8  664.01
  5789.5  663.95    5839   667.5  5846.8  666.25  5888.4  668.87  6089.1  673.79
#Mann= 4 ,-1 , 0
  2564.8      .1       0  4837.1     .12       0  4990.3     .07       0
  5012.3      .1       0
Bank Sta=4990.3,5012.3
XS Rating Curve= 0 ,0
Exp/Cntr=0.3,0.1

Type RM Length L Ch R = 1 ,124817  ,861,861,861
BEGIN DESCRIPTION:
Mapping XS db24f053
END DESCRIPTION:
XS GIS Cut Line= 3
      1977387.12     13582586.03      1976163.16     13581218.84
      1974392.32     13580125.08
#Sta/Elev= 30
  3642.4  653.86  4341.4  646.04    4553  644.59  4792.4  640.44  4947.4  634.91
  4983.3  632.13  4986.3  628.62  4989.4  627.82  5008.7  628.62  5011.7  633.09
  5039.3  633.34  5174.5  634.04  5351.1   633.7  5379.6  630.99  5415.5  634.01
  5561.2  634.65  5629.5   633.9  5914.5  636.57  6051.6  635.44  6539.9  637.47
  6671.2  639.66  6779.9  643.59  6902.9  645.78  7003.3  650.16  7100.4  651.85
  7165.4  654.16  7265.8     655  7317.9  658.57  7342.4  658.72  7558.8  661.76
#Mann= 12 ,-1 , 0
  3642.4     .05       0  4341.4      .1       0    4553     .05       0
  4792.4      .1       0  4986.3     .07       0  5008.7      .1       0
  5039.3     .16       0  5174.5      .1       0  5561.2     .16       0
  5629.5      .1       0  7100.4     .05       0  7342.4      .1       0
Bank Sta=4986.3,5008.7
XS Rating Curve= 0 ,0
Exp/Cntr=0.3,0.1

Type RM Length L Ch R = 1 ,123956  ,942,942,942
BEGIN DESCRIPTION:
Mapping XS 00fb82d4
END DESCRIPTION:
XS GIS Cut Line= 3
      1977986.06     13581713.61      1977022.54     13580932.38
      1974561.61     13580073.01
#Sta/Elev= 30
  3492.8  648.12  4142.8  643.95  4353.1  639.89  4473.1   640.5  4588.1  638.37
  4774.5  638.22  4862.4  636.05  4896.5  633.98  4981.3   631.5  4984.2  628.74
  4987.2  627.94  5006.7  628.74  5012.4  630.88  5027.2  631.62  5100.3  631.02
  5154.3  632.66  5249.7  632.22  5412.6  634.44  5617.6  637.88  5891.8  639.64
  6041.8  639.38    6097  641.09  6118.2  639.77    6166   639.3  6564.4   639.8
    6951  647.68  7107.5     650  7260.2  654.31  7330.4  657.15  7339.9  657.12
#Mann= 10 ,-1 , 0
  3492.8     .05       0  4142.8      .1       0  4896.5     .16       0
  4984.2     .07       0  5006.7     .16       0  5100.3      .1       0
  5412.6     .05       0    6951      .1       0  7260.2     .05       0
  7330.4      .1       0
Bank Sta=4984.2,5006.7
XS Rating Curve= 0 ,0
Exp/Cntr=0.3,0.1

Type RM Length L Ch R = 1 ,123014  ,489,489,489
BEGIN DESCRIPTION:
Black Creek 130.0
END DESCRIPTION:
XS GIS Cut Line= 3
      1978124.97       13579975.      1976644.07     13579995.75
      1974204.85     13580021.79
#Sta/Elev= 30
  3665.7  656.66  3815.7  655.29  4065.7  650.65  4115.7  648.59  4775.8  633.41
  4805.8  631.18  4858.5  630.41  4925.8  629.58  4975.8  631.19  4984.5   626.6
  4987.6   625.8    5007   626.6  5015.8  629.71  5035.8  628.14  5065.4  630.27
  5095.8  631.62  5168.6  631.97  5205.8  631.24  5435.8   636.5  5635.8  638.68
  6045.9  638.73  6085.9  639.82  6155.9  638.42  6425.9  638.75  6856.2   646.2
  7151.5  653.33  7185.9  653.93  7222.4  656.81  7265.9  656.86  7586.1  668.01
#Mann= 9 ,-1 , 0
  3665.7      .1       0  4858.5     .12       0  4984.5     .07       0
    5007     .12       0  5065.4      .1       0  5168.6     .05       0
  6856.2      .1       0  7151.5     .05       0  7222.4      .1       0
Bank Sta=4984.5,5007
XS Rating Curve= 0 ,0
Exp/Cntr=0.3,0.1

Type RM Length L Ch R = 1 ,122525  ,800,800,800
BEGIN DESCRIPTION:
Black Creek 129.0
END DESCRIPTION:
XS GIS Cut Line= 3
       1978131.9     13579575.17        1977059.     13579549.13
      1974600.63     13579632.47
#Sta/Elev= 30
  3778.5  654.63  3955.4  654.22  4095.5  652.72  4225.5  648.71  4345.6  645.96
  4485.6   641.3  4745.7  635.06  4765.7  633.82  4863.5   630.9  4975.8  628.48
  4984.5  625.72  4987.6  624.92    5004  624.92    5007  625.72  5015.8  629.01
  5045.8  628.33  5095.9  628.99  5105.9  629.88  5125.9  629.38  5191.3   630.1
  5235.9  630.36  5486.1  635.79  5636.2  637.19  5896.3  637.67  6316.6  637.07
  6586.7  637.71  6736.8  639.31  7087.7  646.25  7260.5  651.26  7311.5  652.37
#Mann= 7 ,-1 , 0
  3778.5      .1       0  4863.5     .12       0  4984.5     .07       0
    5007     .12       0  5191.3     .05       0  7087.7      .1       0
  7260.5     .05       0
Bank Sta=4984.5,5007
XS Rating Curve= 0 ,0
Exp/Cntr=0.3,0.1

Type RM Length L Ch R = 1 ,121725  ,592,592,592
BEGIN DESCRIPTION:
Mapping XS 73c20d7d
END DESCRIPTION:
XS GIS Cut Line= 4
      1978215.27     13579366.86       1977439.2     13578809.55
      1975345.45     13578960.59      1974225.62     13578684.54
#Sta/Elev= 30
  3524.8  651.43  3827.4  647.26  4177.6  639.47    4364  639.34  4604.8  636.47
  4855.4  631.35  4903.2  628.69  4955.7  627.13  4975.7  627.73  4984.5  624.82
  4987.6  624.02  5007.1  624.82  5015.8  627.26  5025.9  627.64    5086  628.43
  5146.2  627.05  5360.1  632.49  5600.4  635.53  5906.3  635.27  5966.2  634.78
  6118.7  634.68  6509.7  637.63  6734.4   640.7  6956.9  641.55  7418.4  646.83
    7476  649.27  7501.4   648.1  7506.8  649.66  7525.7  649.89  7732.8  653.34
#Mann= 9 ,-1 , 0
  3524.8      .1       0  4903.2     .12       0  4984.5     .07       0
  5007.1     .12       0  5146.2      .1       0  5360.1     .05       0
  5906.3      .1       0  5966.2     .05       0  7525.7      .1       0
Bank Sta=4984.5,5007.1
XS Rating Curve= 0 ,0
Exp/Cntr=0.3,0.1

Type RM Length L Ch R = 1 ,121133  ,964,964,964
BEGIN DESCRIPTION:
Mapping XS 3d7d0d75
END DESCRIPTION:
XS GIS Cut Line= 3
      1978272.55     13578554.34      1976147.54     13578241.84
      1974793.39     13578122.05
#Sta/Elev= 30
  3482.1  647.97  4217.5  637.43  4449.9  636.52  4755.6   632.6  4783.5  632.93
  4975.5   626.1  4984.5  623.12  4987.6  622.32  5007.1  623.12    5016  627.09
  5027.6  627.46  5106.9  627.31  5127.2  623.46  5158.3  626.67    5441  629.31
  5500.6   632.8  5505.7  631.92  5551.7  636.87  5649.2   634.2  5654.2  635.49
  5729.4  634.54  5761.2  634.86  5773.1  636.59  6064.4  640.55  6285.1  644.03
  6596.3  643.45  6616.3  647.93  6626.4  643.97  6646.5  643.43  6989.4  648.43
#Mann= 7 ,-1 , 0
  3482.1      .1       0  4755.6     .12       0  4984.5     .07       0
  5007.1     .12       0  5158.3      .1       0  5729.4     .05       0
  6064.4      .1       0
Bank Sta=4984.5,5007.1
XS Rating Curve= 0 ,0
Exp/Cntr=0.3,0.1

Type RM Length L Ch R = 1 ,120169  ,715,715,715
BEGIN DESCRIPTION:
Mapping XS 753fa435
END DESCRIPTION:
XS GIS Cut Line= 2
      1978074.62     13577856.42      1974976.98     13577309.78
#Sta/Elev= 30
  3371.4  642.56  3787.3  635.26  4530.2  630.49  4620.9  630.31  4691.1  628.55
  4711.4  627.27  4802.8  626.64  4847.7  625.38    4945  624.66  4961.1  626.31
  4975.4  625.71  4984.4  621.87  4987.5  621.07  5003.9  621.07  5007.1  621.87
  5015.3  625.58  5036.4  624.96  5085.7  626.25  5127.7  627.58  5148.1  627.31
  5158.2  628.28  5259.8  628.78  5538.2  633.59  5705.8  639.37  5818.2  641.39
  5824.2  642.43  5858.9  642.47  6102.6  647.54  6342.1  650.05  6516.9  653.06
#Mann= 5 ,-1 , 0
  3371.4      .1       0  4530.2     .12       0  4984.4     .07       0
  5007.1     .12       0  5085.7      .1       0
Bank Sta=4984.4,5007.1
XS Rating Curve= 0 ,0
Exp/Cntr=0.3,0.1

Type RM Length L Ch R = 1 ,119454  ,724,724,724
BEGIN DESCRIPTION:
Mapping XS d9a81639
END DESCRIPTION:
XS GIS Cut Line= 2
      1978100.66     13577439.76      1975179.39     13576455.58
#Sta/Elev= 30
  3375.1  641.42  3747.7  633.76  4077.5  631.33  4362.4  631.22  4682.4  627.96
  4900.6  624.66  4932.3  622.49  4975.7   624.9    4985  622.83  4995.6  622.27
    5002  624.51  5038.7  625.33  5059.4  630.33    5080  626.64  5090.5  623.63
  5096.4  619.93  5101.7     621  5116.6  618.49  5119.7  617.69  5139.3  618.49
  5196.2   623.7  5222.4  623.79  5259.4  627.72  5301.6  628.95  5702.6  636.38
  5757.7  635.94  5972.8  640.92  6067.3  641.53  6408.4  651.33  6457.7  651.72
#Mann= 5 ,-1 , 0
  3375.1      .1       0  4682.4     .12       0  5059.4      .1       0
  5116.6     .07       0  5139.3      .1       0
Bank Sta=5116.6,5139.3
XS Rating Curve= 0 ,0
Exp/Cntr=0.3,0.1

Type RM Length L Ch R = 1 ,118730  ,735,735,735
BEGIN DESCRIPTION:
Black Creek 122.0
END DESCRIPTION:
XS GIS Cut Line= 3
      1978178.76     13577241.82      1976819.41     13576398.09
       1975439.6     13575596.24
#Sta/Elev= 30
  3073.1  640.66  3193.7  638.67    3227  637.93  3310.6  636.27  3430.6  633.26
  3690.1  630.96  3762.6  632.62  3771.9  631.28  3787.1  631.46  4329.5  629.35
  4799.3  625.69  4831.3  625.54  4847.1  623.48  4955.7  622.75  4980.6  620.42
  4983.7  619.62  5003.3  620.42  5013.5  623.33  5029.2  623.81  5221.2  622.99
  5263.2   625.1  5418.3  628.27  5489.4  630.98  5548.1  631.03  5644.2  633.48
  5702.9  633.57  5708.7  632.26  5740.2  634.73  5847.8     635  6268.9  641.28
#Mann= 10 ,-1 , 0
  3073.1     .05       0  3193.7      .1       0    3227     .05       0
  3310.6      .1       0  3690.1     .05       0  3787.1      .1       0
  4799.3     .12       0  4980.6     .07       0  5003.3     .12       0
  5263.2      .1       0
Bank Sta=4980.6,5003.3
XS Rating Curve= 0 ,0
Exp/Cntr=0.3,0.1

Type RM Length L Ch R = 1 ,117995  ,649,649,649
BEGIN DESCRIPTION:
Black Creek 124.0
END DESCRIPTION:
XS GIS Cut Line= 3
      1978319.43     13577064.77       1977001.7     13575866.84
      1975851.81     13574899.06
#Sta/Elev= 30
  2808.5  636.19  3007.5  636.44  3179.4  635.62  3385.6     632  3514.8  629.83
  3710.1  629.36  3773.3   629.4  3902.6  629.52  4031.8  628.85    4161  629.09
  4453.5  628.87  4675.3  626.62    4796  623.71  4925.8     623  5122.9  620.91
  5126.1  620.11  5145.6  620.91  5269.5  622.75    5286   624.7  5462.1  628.28
  5552.1  630.64  5595.9  630.21  5638.8  632.86  5786.8  635.98  5957.5  639.82
  5979.6   644.5  6022.5  643.73  6035.9  645.28  6052.7  643.44  6092.3  643.08
#Mann= 20 ,-1 , 0
  2808.5      .1       0  3007.5      .1       0  3385.6     .05       0
  3514.8     .08       0  3710.1      .1       0  3773.3     .08       0
  3902.6     .08       0  4031.8     .08       0    4161     .05       0
  4453.5      .1       0  4675.3      .1       0    4796     .08       0
  4925.8     .12       0  5122.9     .07       0  5145.6     .08       0
    5286     .08       0  5462.1      .1       0  5552.1     .05       0
  5786.8     .08       0  6052.7      .1       0
Bank Sta=5122.9,5145.6
XS Rating Curve= 0 ,0
Exp/Cntr=0.3,0.1

Type RM Length L Ch R = 1 ,117346  ,603,603,603
BEGIN DESCRIPTION:
Black Creek 123.0
END DESCRIPTION:
XS GIS Cut Line= 3
      1979751.74     13577377.29      1977069.41      13575153.3
      1976272.56     13574450.19
#Sta/Elev= 30
  1453.7  636.17  1481.4  636.64  1558.5  634.57  1717.8   633.3  1718.9  633.29
  2071.3  632.79  2439.9  634.11  2883.1  629.56  2963.8  628.33  3025.4  628.47
  3090.5  628.51  3360.7  628.75  3437.3  628.91    3782  628.96  4578.3  626.08
  4769.7  621.34  4918.1     621  4932.5  618.73  4968.6  621.59  4975.3  621.17
  4985.7   615.1  4988.9   614.3  5008.5   615.1  5010.7  619.13    5018  619.59
  5181.1  625.38  5308.3  626.11  5365.2  627.71    5627  628.31  6000.8  634.78
#Mann= 13 ,-1 , 0
  1453.7      .1       0  1558.5     .05       0  1717.8      .1       0
  1718.9     .05       0  2883.1      .1       0  2963.8     .05       0
  3025.4      .1       0  3090.5     .05       0  3360.7      .1       0
  3437.3     .05       0    3782      .1       0  4985.7     .07       0
  5008.5      .1       0
Bank Sta=4985.7,5008.5
XS Rating Curve= 0 ,0
Exp/Cntr=0.3,0.1

Type RM Length L Ch R = 1 ,116743  ,757,757,757
BEGIN DESCRIPTION:
Mapping XS b8e5b598
END DESCRIPTION:
XS GIS Cut Line= 3
      1978801.22     13575347.76      1977377.57     13574823.44
      1976239.34     13574382.72
#Sta/Elev= 30
  3579.7  637.65  4093.3  628.13  4364.3  625.14  4480.1  624.92    4652  622.78
  4772.4  623.43  4792.2  623.89  4872.9  619.22  4964.2  620.15  4982.3  619.59
  4983.2  615.74  4986.4  614.94  5002.9  614.94  5006.1  615.74  5014.3  619.94
  5025.1  620.27  5044.9  619.38  5080.7  620.49    5111  619.64  5142.5  620.46
  5160.2  618.66  5174.7  619.88  5228.3  621.73    5239  621.33  5266.8  622.99
  5383.9   624.3  5614.3  627.95  5988.4  629.68  6202.3  633.41  6317.4   635.4
#Mann= 8 ,-1 , 0
  3579.7     .05       0  4480.1      .1       0  4772.4     .16       0
  4983.2     .07       0  5006.1     .16       0  5266.8      .1       0
  5383.9     .05       0  6202.3      .1       0
Bank Sta=4983.2,5006.1
XS Rating Curve= 0 ,0
Exp/Cntr=0.3,0.1

Type RM Length L Ch R = 1 ,115986  ,560,560,560
BEGIN DESCRIPTION:
Black Creek 121.0
END DESCRIPTION:
XS GIS Cut Line= 4
      1979183.97     13574684.54      1978631.91     13574507.47
       1977371.5     13574293.92      1976204.81     13574330.38
#Sta/Elev= 30
  3616.5  641.66  4289.4  630.68  4548.1  626.09    4609  624.15  4639.4  624.95
  4717.7  622.13  4832.1  621.18  4898.8  618.73  4964.2  618.24  4982.9  615.87
  4986.1  615.07  5005.8  615.87  5014.4  617.34  5041.5  617.94  5074.8  618.03
  5079.8  616.44  5085.7  616.33  5095.8  618.06  5142.9  618.03  5217.5  620.12
  5349.4  621.91  5410.2   624.1    5442  622.29  5450.8  622.58  5470.3  626.71
  5537.9  627.11  5841.3  629.74  6331.6  630.84  6609.5  634.88  6641.9  635.45
#Mann= 8 ,-1 , 0
  3616.5     .05       0  4289.4      .1       0  4982.9     .07       0
  5005.8      .1       0  5041.5     .16       0  5142.9      .1       0
  5537.9     .05       0  6609.5      .1       0
Bank Sta=4982.9,5005.8
XS Rating Curve= 0 ,0
Exp/Cntr=0.3,0.1

Type RM Length L Ch R = 1 ,115426  ,636,636,636
BEGIN DESCRIPTION:
Black Creek 120.0
END DESCRIPTION:
XS GIS Cut Line= 4
      1978907.96     13573918.93      1978642.33     13573799.13
      1977423.58     13573918.92      1976272.55     13574273.09
#Sta/Elev= 30
  3906.3  634.04  4146.2  633.98  4225.2  632.06  4325.6  627.63  4416.1  625.53
  4661.5  623.18  4862.3  618.61  4922.8  617.37  4948.6  617.72  4961.5  616.82
  4978.8  616.77  4987.4  613.05  4990.6  612.25  5007.1  612.25  5010.4  613.05
    5019  616.67  5060.6  617.05  5099.4  615.71  5159.8  617.77  5260.1  619.19
  5350.6  623.81  5380.7  624.29  5400.8  627.01  5443.4  627.57  5535.9  628.02
  5567.3  626.85  5660.1  626.92  5866.8     628  6378.1  631.08  6626.6  634.09
#Mann= 9 ,-1 , 0
  3906.3     .05       0  4661.5      .1       0  4862.3     .07       0
  4961.5     .16       0  4987.4     .07       0  5010.4     .16       0
  5060.6     .12       0  5159.8      .1       0  5443.4     .05       0
Bank Sta=4987.4,5010.4
XS Rating Curve= 0 ,0
Exp/Cntr=0.3,0.1

Type RM Length L Ch R = 1 ,114790  ,562,562,562
BEGIN DESCRIPTION:
Black Creek 119.0
END DESCRIPTION:
XS GIS Cut Line= 4
      1979092.87     13573434.55      1978363.68     13573247.05
      1977113.68     13573517.88      1976117.12     13574191.52
#Sta/Elev= 30
  3497.2  636.99  3587.9  636.79  3716.6  634.55    3939  627.83  4062.9  625.33
  4320.4  622.86  4629.4  622.18  4719.4  621.08  4839.2  616.86  4883.1  615.95
  4954.5  616.08  4976.4  616.15    5009  612.63  5012.2  611.83  5028.7  611.83
    5032  612.63  5036.6  614.04  5069.7  616.43  5108.3  617.63  5113.7  616.72
  5118.8  617.95  5128.7   616.9  5142.7  616.84  5212.1  619.62  5282.2  620.08
  5548.2  624.75  5648.2  625.23  5937.7  628.75  6390.3  631.56    6732  635.66
#Mann= 7 ,-1 , 0
  3497.2     .05       0  4629.4      .1       0  4839.2     .12       0
  4954.5      .1       0    5009     .07       0    5032      .1       0
  5142.7     .05       0
Bank Sta=5009,5032
XS Rating Curve= 0 ,0
Exp/Cntr=0.3,0.1

Type RM Length L Ch R = 1 ,114228  ,551,551,551
BEGIN DESCRIPTION:
Black Creek 118.0
END DESCRIPTION:
XS GIS Cut Line= 4
      1979273.38     13573031.76      1978526.24     13572671.66
      1977023.41     13572983.16      1976120.65     13573795.64
#Sta/Elev= 30
  3100.3     637  3253.9   635.3  3509.2  630.69    3809   626.6  4237.3  622.32
  4471.3  621.87  4615.8  621.64  4685.7  620.17  4718.9   619.3  4788.8  616.01
  4850.1  614.41  4911.7  615.68  4972.6  615.55  4982.9  614.79  4990.3  612.53
  4993.6  611.73  5010.1  611.73  5013.3  612.53  5013.5  614.42  5031.8   615.6
  5064.6  618.69  5207.6  619.39  5340.3  621.46    5507  627.04  5641.5  629.55
  5875.5  630.18  5924.8  629.49  6144.6   629.4  6420.4  630.19    6679   634.5
#Mann= 7 ,-1 , 0
  3100.3     .05       0  4471.3      .1       0  4685.7     .16       0
  4718.9      .1       0  4990.3     .07       0  5013.3      .1       0
  5031.8     .05       0
Bank Sta=4990.3,5013.3
XS Rating Curve= 0 ,0
Exp/Cntr=0.3,0.1

Type RM Length L Ch R = 1 ,113677  ,714,714,714
BEGIN DESCRIPTION:
Black Creek 117.0
END DESCRIPTION:
XS GIS Cut Line= 4
      1979502.55      13572302.6      1978363.68      13572240.1
      1977002.57      13572427.6      1976092.85     13573573.44
#Sta/Elev= 30
  3028.3  648.53  3246.2  641.88  3266.2  640.08  3276.2  640.22  3296.3  643.75
  3306.3  643.49  3316.3  641.05  3336.3  639.16  3606.7  632.27  4177.6  624.58
  4369.4   623.8  4409.8  622.19  4756.5  618.62  4904.1  616.04    4965  613.08
  4972.1  610.84  4983.7  609.74    4987  608.94  5006.8  609.74  5035.7   613.8
  5103.5  614.36  5203.3  617.22    5486   619.9  5724.3  619.54  5809.2  621.96
    5846  621.67  5881.3   623.2  6158.5  627.63  6599.3  628.58  7005.9  632.86
#Mann= 7 ,-1 , 0
  3028.3     .05       0  4756.5      .1       0  4904.1     .12       0
  4983.7     .07       0  5006.8     .12       0  5103.5      .1       0
  5203.3     .05       0
Bank Sta=4983.7,5006.8
XS Rating Curve= 0 ,0
Exp/Cntr=0.3,0.1

Type RM Length L Ch R = 1 ,112963  ,903,903,903
BEGIN DESCRIPTION:
Black Creek 116.0
END DESCRIPTION:
XS GIS Cut Line= 3
      1979238.73     13571233.15      1977134.52      13571821.7
      1975973.03     13572764.44
#Sta/Elev= 30
  3112.3  639.23    3490  634.91    3885  627.73  4081.9  626.46    4213   624.3
  4299.9  624.71  4351.8  622.48    4653  618.45  4781.2  615.55    4871  613.52
  4928.8  613.66  4985.3  612.67  4985.8  610.47  4989.1  609.67  5005.6  609.67
  5008.9  610.47  5016.4  612.38  5046.3  611.98    5105  615.06  5172.2  615.63
  5426.7     622    5676  624.21  5789.5     623    5847  623.76    6237  624.16
  6443.2  626.36  6649.4  630.89  6686.1  630.41  6692.5  629.48  6793.2  631.12
#Mann= 6 ,-1 , 0
  3112.3     .05       0  4781.2      .1       0  4928.8     .12       0
  4985.8     .07       0  5008.9     .12       0  5046.3     .05       0
Bank Sta=4985.8,5008.9
XS Rating Curve= 0 ,0
Exp/Cntr=0.3,0.1

Type RM Length L Ch R = 1 ,112060  ,669,669,669
BEGIN DESCRIPTION:
Black Creek 115.0
END DESCRIPTION:
XS GIS Cut Line= 3
      1978426.21     13570113.36      1977160.56     13570774.83
      1975947.02     13572238.37
#Sta/Elev= 30
  3144.7  676.44  3183.1  675.45  3309.9  662.79  3399.6  658.76  3518.4  652.72
  3525.1  653.09  3530.7  651.89  3574.9   649.9  3657.5  647.26  3679.6  645.28
  3732.8  642.77  3955.3  634.65  4037.4  632.74  4286.5  623.58  4566.6  617.14
  4839.6  613.41  4874.8  610.91  4920.6   609.6  4923.9   608.8  4940.4   608.8
  4943.7   609.6  4981.6  610.08  5080.6  614.75  5117.1  614.68  5152.2  616.23
  5393.1  616.21    5621  621.93  5656.2  621.27  6182.3  623.26    6474  628.89
#Mann= 5 ,-1 , 0
  3144.7      .1       0  3399.6     .05       0  4566.6      .1       0
  4920.6    .035       0  4943.7     .05       0
Bank Sta=4920.6,4943.7
XS Rating Curve= 0 ,0
Exp/Cntr=0.3,0.1

Type RM Length L Ch R = 1 ,111391  ,859,859,859
BEGIN DESCRIPTION:
Black Creek 114.0
END DESCRIPTION:
XS GIS Cut Line= 3
      1977975.02     13569474.98        1976425.       13570625.
      1975811.62     13571748.74
#Sta/Elev= 30
  3064.1  671.53    3087  669.65  3113.9  667.37  3136.1  663.72  3171.6  659.62
  3250.9  655.95  3350.5  649.43  3672.4   635.7  3899.7  629.11  3979.1   628.5
  4058.4  626.05  4229.5  622.88  4271.9  622.94  4612.3   616.2  4794.9  613.97
  4857.5  614.57  4922.1     610  4972.7  608.06  4975.2  607.63  4978.6  606.83
  4998.4  607.63  5051.6  611.02  5089.5  610.93    5378  617.42  5383.7  616.44
    5547  619.46  5835.5  621.16    6032   620.6  6189.5  622.51  6274.4  622.41
#Mann= 6 ,-1 , 0
  3064.1      .1       0    3087     .05       0  4612.3      .1       0
  4972.7     .05       0  4975.2    .035       0  4998.4     .05       0
Bank Sta=4975.2,4998.4
XS Rating Curve= 0 ,0
Exp/Cntr=0.3,0.1

Type RM Length L Ch R = 1 ,110532  ,386,386,386
BEGIN DESCRIPTION:
Black Creek 113.0
END DESCRIPTION:
XS GIS Cut Line= 3
      1976925.02     13569374.99      1975737.82     13570062.15
      1975758.65     13571249.64
#Sta/Elev= 30
  4077.5  639.22  4261.9  631.26  4283.4  629.96  4422.6  625.11  4471.5   622.8
  4539.7  621.12  4604.9   618.7  4706.8  616.22  4787.1  613.35  4824.4  611.55
  4920.6  610.29  4963.6  609.13  4978.8  609.28  4985.2  608.69  4989.3  605.55
  4992.7  604.75  5009.2  604.75  5012.5  605.55  5013.4  607.92  5022.5  608.92
    5044  608.67  5094.3  609.52  5152.1  611.39    5189  611.98  5343.9  612.65
  5542.1   614.5  5552.1  615.03  5902.1  615.67  6412.2  619.65  6636.9  620.41
#Mann= 3 ,-1 , 0
  4077.5     .05       0  4989.3    .035       0  5012.5     .05       0
Bank Sta=4989.3,5012.5
XS Rating Curve= 0 ,0
Exp/Cntr=0.3,0.1

Type RM Length L Ch R = 1 ,110146  ,471,471,471
BEGIN DESCRIPTION:
Black Creek 112.0
END DESCRIPTION:
XS GIS Cut Line= 4
       1976740.3     13569219.42      1975818.41     13569542.34
      1975141.32     13569630.88       1973839.6     13569464.26
#Sta/Elev= 30
  4163.7  639.08  4264.7  633.47  4785.7  612.47  4932.2  609.05    4950  607.41
  4955.3  608.43    4981  608.18  4984.2  605.41  4987.5  604.61  5007.4  605.41
  5012.1  607.73  5042.2  608.33  5099.8  608.97    5154  611.47  5345.6   613.5
  5547.4  611.67  5759.1  612.02  5897.6  610.69  5940.6  609.82  5970.9  606.74
  5986.9  609.36  6051.5  610.11  6539.8  618.42    6727  623.03  6747.2  624.98
  6787.5   625.5  6837.9   628.3  6853.6  626.66  6908.5  627.31  7135.7  634.83
#Mann= 7 ,-1 , 0
  4163.7     .05       0  4785.7      .1       0  4984.2     .07       0
  5007.4      .1       0  5042.2     .05       0  5897.6      .1       0
  6051.5     .05       0
Bank Sta=4984.2,5007.4
XS Rating Curve= 0 ,0
Exp/Cntr=0.3,0.1

Type RM Length L Ch R = 1 ,109675  ,697,697,697
BEGIN DESCRIPTION:
Black Creek 111.0
END DESCRIPTION:
XS GIS Cut Line= 3
      1976823.61     13568927.76      1975349.66     13569229.84
      1973860.05     13569235.05
#Sta/Elev= 30
  3779.3  643.49  3892.7  640.42  3988.4  636.54  4084.1  634.41  4451.6  619.51
  4690.4  612.27  4767.8  610.65  4848.5  609.47  4972.2  608.25  4981.6  607.72
  4991.2   604.8  4994.5     604  5014.4   604.8  5023.2  606.74    5071  608.06
  5137.9  610.35  5370.2     611  5498.5  609.53  5568.5   605.5  5578.5  605.64
  5588.5  607.86  5598.5  608.52    5669  609.43  5888.5  612.38  6138.5  618.93
  6388.5  629.06  6428.5  631.61  6468.5  632.46  6628.6   640.3  6773.5   643.4
#Mann= 9 ,-1 , 0
  3779.3     .05       0  4690.4      .1       0  4767.8     .05       0
  4848.5      .1       0  4991.2     .07       0  5014.4      .1       0
    5071     .05       0  5370.2      .1       0    5669     .05       0
Bank Sta=4991.2,5014.4
XS Rating Curve= 0 ,0
Exp/Cntr=0.3,0.1

Type RM Length L Ch R = 1 ,108978  ,259,259,259
BEGIN DESCRIPTION:
Black Creek 110.0
END DESCRIPTION:
XS GIS Cut Line= 3
      1977302.82     13568682.97      1975193.41     13568677.76
      1974101.15      13568870.2
#Sta/Elev= 30
  2830.6  645.78  3068.4  635.82  3118.4  634.65  3308.4  635.31  3368.4  634.57
  3558.4   629.1  3738.4  626.04  3978.4  619.96  4328.4  614.44  4706.2  610.05
  4818.4  607.26  4928.4  607.94  4968.9  607.36  4976.9  605.07  4980.7  604.27
  4997.6  604.27  5001.5  605.07  5007.5  607.07  5039.9  605.64  5080.6  607.27
  5101.1  606.99  5364.9  610.67  5530.8  615.24    5639  619.89  5762.9  626.56
  5817.1  630.69  5876.3  633.87  5930.5  638.86    5964  640.55  6049.1  642.58
#Mann= 5 ,-1 , 0
  2830.6     .05       0  4706.2      .1       0  4976.9     .07       0
  5001.5      .1       0  5101.1     .05       0
Bank Sta=4976.9,5001.5
XS Rating Curve= 0 ,0
Exp/Cntr=0.3,0.1

Type RM Length L Ch R = 1 ,108719  ,392,392,392
BEGIN DESCRIPTION:
Black Creek 109.0
END DESCRIPTION:
XS GIS Cut Line= 3
      1977344.41     13567667.35        1974975.       13568475.
      1974110.09     13568776.71
#Sta/Elev= 30
    2526  638.83  2657.8  637.33  2877.2  637.09  2958.5  636.16  3305.5  636.77
  3373.5  634.38  3613.6  630.06  4052.5  616.64  4172.6  614.12  4479.9  611.96
  4770.9  608.03  4870.8  606.36  4982.3  606.83  4985.3     604  4989.1   603.2
    5006   603.2  5009.9     604  5013.6  606.16  5044.8  605.83  5052.9  606.68
  5070.6  607.71  5124.6  607.78  5325.8  611.83  5500.2  617.98  5624.5  623.96
  5681.3  628.36  5743.5  631.54  5844.8  638.48  5876.6  639.96  5945.3   641.1
#Mann= 5 ,-1 , 0
    2526     .05       0  4770.9      .1       0  4985.3     .07       0
  5009.9      .1       0  5052.9     .05       0
Bank Sta=4985.3,5009.9
XS Rating Curve= 0 ,0
Exp/Cntr=0.3,0.1

Type RM Length L Ch R = 1 ,108327  ,621,621,621
BEGIN DESCRIPTION:
Black Creek 108.0
END DESCRIPTION:
XS GIS Cut Line= 4
        1976225.       13567975.      1975516.32      13567891.3
      1974641.32     13568245.46      1974174.97     13568725.03
#Sta/Elev= 30
    3744  628.94  3985.7  623.05  4124.6  616.66  4267.6  612.46  4418.7  610.44
  4801.7   608.4    4869   607.3  4882.9  607.99  4890.6  609.28    4907  609.99
  4990.1   605.1  5030.8  606.26  5043.7  605.27  5067.9  606.02  5106.3  605.38
  5115.6  604.67  5119.4  603.87  5136.3  603.87  5140.2  604.67  5145.6  606.71
    5151  607.04  5160.3  606.67  5199.4  607.46  5235.8  607.71    5434  613.79
  5575.4  616.46  5681.4  619.78    5731  620.66  5964.4  634.07  6070.5  639.23
#Mann= 5 ,-1 , 0
    3744     .05       0  4801.7      .1       0  5115.6     .07       0
  5140.2      .1       0  5199.4     .05       0
Bank Sta=5115.6,5140.2
XS Rating Curve= 0 ,0
Exp/Cntr=0.3,0.1

Type RM Length L Ch R = 1 ,107706  ,714,714,714
BEGIN DESCRIPTION:
Black Creek 107.0
END DESCRIPTION:
XS GIS Cut Line= 3
      1977183.01     13567370.46       1975063.2     13567531.92
      1974011.45     13567610.02
#Sta/Elev= 30
  2696.3  631.13  2776.5  630.15  2875.4  628.86  3082.8  627.74  3165.7  628.99
  3369.9  625.79    3978  619.07  4098.4  614.17    4267  610.59  4583.9  608.33
  4655.4  607.78  4750.2  608.06  4853.1  605.61  4920.7  603.39  4960.8  604.94
  4970.9  604.37  4978.5  599.83  4982.4  599.03  5003.4  599.83    5011   604.7
  5050.8  605.51  5121.3  607.33  5281.7  606.55  5354.5   609.1  5513.2  614.43
  5582.5  614.99    5644  617.81  5692.8  618.61  5743.2  621.89  5876.9  626.75
#Mann= 14 ,-1 , 0
  2696.3     .05       0  2776.5     .08       0  2875.4      .1       0
  3369.9     .05       0  4583.9     .08       0  4655.4     .05       0
  4853.1     .12       0  4978.5     .07       0  5003.4     .12       0
  5050.8     .16       0  5354.5      .1       0  5513.2     .08       0
    5644     .05       0  5743.2      .1       0
Bank Sta=4978.5,5003.4
XS Rating Curve= 0 ,0
Exp/Cntr=0.3,0.1

Type RM Length L Ch R = 1 ,106992  ,689,689,689
BEGIN DESCRIPTION:
Black Creek 106.0
END DESCRIPTION:
XS GIS Cut Line= 3
      1976995.51      13566703.8        1974825.       13566875.
        1973584.     13566912.13
#Sta/Elev= 30
  2838.6  630.31  3079.9   629.2  3812.4  619.46  3972.6  618.08  3992.7  618.56
  4032.8  617.09  4153.2  615.01  4373.9  608.78  4673.3  607.28  4815.2  606.21
  4855.4  604.14  4885.4  605.49  4945.6  602.92  4956.5  603.36  4975.7  602.57
  4983.3  599.17  4987.3  598.37  5004.3  598.37  5008.2  599.17  5013.3  603.43
  5095.9   602.2  5114.9  602.78  5175.9  604.16    5266  608.23  5498.2  615.37
  5526.1  617.26  5626.1  619.96  5856.5  629.84  6106.3   630.9  6257.4  634.69
#Mann= 6 ,-1 , 0
  2838.6     .05       0  4673.3     .16       0  4983.3     .07       0
  5008.2     .16       0  5114.9      .1       0  5498.2     .05       0
Bank Sta=4983.3,5008.2
XS Rating Curve= 0 ,0
Exp/Cntr=0.3,0.1

Type RM Length L Ch R = 1 ,106303  ,1095,1095,1095
BEGIN DESCRIPTION:
Mapping XS 794d57eb
END DESCRIPTION:
XS GIS Cut Line= 3
      1977016.32     13566406.92      1975781.95     13566057.96
      1973408.52     13566536.81
#Sta/Elev= 30
  2512.3  626.09  2617.6   624.3  2731.9  624.74  2977.5  622.49  3729.5  613.32
    3852   612.9  4055.1  615.07  4212.6  614.17  4469.3  608.42    4563   607.6
  4699.9  604.57  4838.3  604.77  4913.4  601.74  4944.7  601.91  4964.2  604.18
  4985.5  601.55  4993.5  596.73  4997.4  595.93  5018.4  596.73  5026.3  601.88
  5036.5  602.41  5116.5  602.47  5223.8  606.51  5301.8  608.48  5324.8  610.07
  5527.9  612.99  5827.5  623.57  6030.7  627.59  6158.7  631.92  6216.3  632.33
#Mann= 6 ,-1 , 0
  2512.3     .05       0  4469.3      .1       0  4838.3     .16       0
  4993.5     .07       0  5018.4     .16       0  5223.8     .05       0
Bank Sta=4993.5,5018.4
XS Rating Curve= 0 ,0
Exp/Cntr=0.3,0.1

Type RM Length L Ch R = 1 ,105208  ,447,447,447
BEGIN DESCRIPTION:
Black Creek 105.0
END DESCRIPTION:
XS GIS Cut Line= 3
      1977026.78     13565990.27        1974475.       13565325.
      1973059.02     13565391.25
#Sta/Elev= 30
  2375.5  622.74  2672.7  618.68  2821.7  616.68  2890.4  617.39  3638.1  610.99
  4160.2  609.54  4165.3   608.6  4206.5  608.84  4241.1  607.07  4357.4  604.99
  4362.6  606.75  4366.8  606.62  4423.5  603.71  4514.2  603.22  4702.5  605.06
  4830.6  603.03  4878.6  603.06  4929.9  599.49  4971.2  600.35  4977.2  595.99
  4981.2  595.19  5002.2  595.99    5010  599.56  5042.6  599.19    5176  603.72
  5262.8  605.63  5453.1  606.75  5743.4  611.75  6023.7  612.68  6430.1  617.47
#Mann= 7 ,-1 , 0
  2375.5     .12       0  2672.7     .05       0  4366.8      .1       0
  4830.6     .16       0  4977.2     .07       0  5002.2     .16       0
    5176      .1       0
Bank Sta=4977.2,5002.2
XS Rating Curve= 0 ,0
Exp/Cntr=0.3,0.1

Type RM Length L Ch R = 1 ,104761  ,164,164,164
BEGIN DESCRIPTION:
Black Creek 104.0
END DESCRIPTION:
XS GIS Cut Line= 3
       1977125.7     13564776.71      1974703.82     13564917.34
       1973203.8     13565011.09
#Sta/Elev= 30
  2460.8   620.8  2697.6  617.99  2852.3  616.73    2895   616.5    3379  612.66
  3980.8  611.49  4174.2  611.89  4304.6  610.05    4515  602.05  4575.1  601.87
  4655.2  603.57  4770.5  603.17  4886.8  601.63  4935.7  598.78  4965.7  599.55
  4967.9  598.71  4973.3  596.65  4977.3  595.85  4998.3  596.65  5005.8  599.96
  5046.6  599.34  5090.3  599.62  5156.1  603.39  5374.2  605.15  5647.1     607
  6052.2   614.4    6138  617.07  6158.1  616.23  6298.3  616.66  6389.7  618.06
#Mann= 12 ,-1 , 0
  2460.8     .05       0  2697.6      .1       0  2852.3     .08       0
    2895     .05       0  3980.8      .1       0  4174.2     .05       0
  4770.5     .08       0  4967.9     .05       0  4973.3     .04       0
  4998.3     .05       0  5046.6     .16       0  5374.2      .1       0
Bank Sta=4973.3,4998.3
XS Rating Curve= 0 ,0
Exp/Cntr=0.3,0.1

Type RM Length L Ch R = 1 ,104597  ,739,739,739
BEGIN DESCRIPTION:
Black Creek 103.0
END DESCRIPTION:
XS GIS Cut Line= 3
      1977219.47     13564615.26      1974620.49     13564776.71
      1973168.64     13564901.61
#Sta/Elev= 30
  2404.7  624.77  2950.2   616.6  3286.7  613.27  3769.1   611.1  4152.5  610.77
  4342.9  609.71  4410.8  608.09  4537.1  603.03  4663.5  601.24  4783.7  603.33
  4843.9  602.95    4903  600.07  4974.1  598.99  4981.6  596.48  4985.6  595.68
  5006.6  596.48  5008.7  598.12  5014.2  599.45  5084.5  599.16  5131.8  602.28
  5161.7  603.54  5244.8  603.29  5375.5  603.97  5385.6  603.03  5556.2  604.82
  5981.6  613.41  6168.4  619.01    6289  619.56  6314.2  619.79  6465.9  620.25
#Mann= 10 ,-1 , 0
  2404.7     .05       0  4410.8      .1       0  4537.1     .05       0
    4903     .16       0  4981.6     .07       0  5006.6     .16       0
  5131.8      .1       0  5244.8     .05       0    6289      .1       0
  6314.2     .05       0
Bank Sta=4981.6,5006.6
XS Rating Curve= 0 ,0
Exp/Cntr=0.3,0.1

Type RM Length L Ch R = 1 ,103858  ,786,786,786
BEGIN DESCRIPTION:
Black Creek 102.0
END DESCRIPTION:
XS GIS Cut Line= 3
      1977255.88     13564151.71      1974943.41     13564084.01
      1973085.76     13564110.02
#Sta/Elev= 30
  2453.9  624.37  2614.9  621.66  2654.9  621.78  2704.9  620.24    2865  617.94
  3365.2  611.74  3995.4  609.32  4668.2  602.65  4715.8  600.94  4766.5  600.99
  4855.8  598.97  4955.8  597.57  4965.8  596.84  4973.2  593.01  4977.2  592.21
  4994.3  592.21  4998.4  593.01  5005.8  596.28  5015.8  597.27  5105.8  601.91
  5145.8  602.62  5334.6  601.42  5506.6  601.44  5575.9  602.46  5595.9  603.71
  5695.9  604.35  5775.9  606.03  5835.9  605.96  6295.9   613.6  6625.2  616.31
#Mann= 8 ,-1 , 0
  2453.9     .05       0  4668.2      .1       0  4766.5     .16       0
  4855.8      .1       0  4973.2     .07       0  4998.4      .1       0
  5334.6      .1       0  5506.6     .05       0
Bank Sta=4973.2,4998.4
XS Rating Curve= 0 ,0
Exp/Cntr=0.3,0.1

Type RM Length L Ch R = 1 ,103072  ,763,763,763
BEGIN DESCRIPTION:
Black Creek 101.0
END DESCRIPTION:
XS GIS Cut Line= 3
      1977531.93     13563380.88        1974425.     13563483.33
      1973124.98     13563533.33
#Sta/Elev= 30
    2196  617.88  2463.1  614.06  2513.1   614.8  2533.1  613.52  2621.1  612.72
  2903.3  609.43  3213.5  607.82  3687.5  610.03  4033.9  610.13  4334.1  605.27
  4394.1  602.59  4583.3  601.09  4681.8   601.1  4794.3  599.95  4834.4  597.58
  4954.4  597.23  4974.4   596.4  4981.8  591.15  4985.9  590.35    5007  591.15
  5014.5  596.57  5084.5  597.96  5114.5  599.66  5443.3   600.2  5544.2  601.11
  5739.1  603.94  6053.4  610.68  6465.5  619.46  6519.7  618.81  6605.6  619.82
#Mann= 9 ,-1 , 0
    2196      .1       0  2621.1     .05       0  4583.3      .1       0
  4681.8     .16       0  4981.8     .07       0    5007     .16       0
  5443.3      .1       0  5544.2     .05       0  6053.4      .1       0
Bank Sta=4981.8,5007
XS Rating Curve= 0 ,0
Exp/Cntr=0.3,0.1

Type RM Length L Ch R = 1 ,102309  ,628,628,628
BEGIN DESCRIPTION:
Black Creek 100.0
END DESCRIPTION:
XS GIS Cut Line= 3
      1977735.12     13562807.97        1974625.       13562725.
      1973174.97     13563075.01
#Sta/Elev= 30
    1897  616.58  2447.3  610.85  2507.3  611.57  2607.4  609.84  2648.4  610.88
  2837.5  607.26  3107.6  605.32  3897.8  606.18  4087.9  604.95    4388  599.48
  4646.3  598.47  4712.2  598.76  4738.1  599.39  4888.2  595.84  4968.2  596.05
  4975.6   591.8  4979.7     591  5000.8   591.8  5005.7  594.38  5018.5  596.25
  5073.6  594.92  5105.2  596.65  5183.1  599.99  5275.7  598.35  5399.1  598.56
  5564.3  601.91  5594.6  602.49  5615.2  605.06  5748.9  607.02  6499.9  628.87
#Mann= 8 ,-1 , 0
    1897      .1       0  2648.4     .05       0  4646.3      .1       0
  4712.2     .16       0  4975.6     .07       0  5000.8     .16       0
  5105.2      .1       0  5564.3     .05       0
Bank Sta=4975.6,5000.8
XS Rating Curve= 0 ,0
Exp/Cntr=0.3,0.1

Type RM Length L Ch R = 1 ,101681  ,193,193,193
BEGIN DESCRIPTION:
Black Creek 99.0
END DESCRIPTION:
XS GIS Cut Line= 4
      1977688.16     13561922.55      1975240.28     13562073.59
      1973615.28     13562198.59      1973069.23      13562302.6
#Sta/Elev= 30
  1976.3  629.09  2257.3  621.35  2652.7  612.75  2851.1  609.41  3191.8  606.53
  3472.3  602.67    3853  602.64  4093.5  603.85  4208.4  603.11  4444.2  598.61
  4662.8  598.64  4846.7  596.33    4902  596.53  4965.7   594.3  4975.7  594.72
  4983.1  592.45  4987.2  591.65  5008.4  592.45  5025.9  595.56  5096.1  594.62
  5162.8  598.56  5228.9  599.11  5346.8  597.57  5497.3  597.46    5644  599.86
  5667.8  600.38  5684.3  602.14  5950.1  605.95  6278.9  614.02  6614.5  618.83
#Mann= 8 ,-1 , 0
  1976.3      .1       0  2652.7     .05       0  4662.8      .1       0
  4846.7     .16       0  4983.1     .07       0  5008.4     .16       0
  5228.9      .1       0    5644     .05       0
Bank Sta=4983.1,5008.4
XS Rating Curve= 0 ,0
Exp/Cntr=0.3,0.1

Type RM Length L Ch R = 1 ,101488  ,829,829,829
BEGIN DESCRIPTION:
Black Creek 98.0
END DESCRIPTION:
XS GIS Cut Line= 3
      1977646.55     13561709.01      1974542.37     13561948.59
      1972891.34     13561995.46
#Sta/Elev= 30
  1972.7  627.31  2112.6  622.63  2445.6  615.63  2927.1  608.36  2957.2  608.74
  3378.4  603.57  3669.3  601.49  3869.9  601.08  4210.9  602.23  4411.5  598.12
    4592  597.67  4662.2  598.41  4692.3  597.14  4713.3  598.28  4812.2  596.49
  4852.8  596.69    4923  594.62  4983.2  595.39  4990.6  593.22  4994.7  592.42
  5011.8  592.42  5015.9  593.22  5023.3  594.28  5053.4  593.51  5103.5  596.63
  5183.5  598.41  5293.6  597.22  5404.9   597.8    6304  613.11  6737.8  618.19
#Mann= 6 ,-1 , 0
  1972.7     .05       0  4713.3     .16       0  4812.2      .1       0
  4990.6     .07       0  5015.9      .1       0  5404.9     .05       0
Bank Sta=4990.6,5015.9
XS Rating Curve= 0 ,0
Exp/Cntr=0.3,0.1

Type RM Length L Ch R = 1 ,100659  ,586,586,586
BEGIN DESCRIPTION:
Black Creek 97.0
END DESCRIPTION:
XS GIS Cut Line= 3
       1977547.6     13561219.42        1974475.       13561175.
       1972729.9     13561255.88
#Sta/Elev= 30
  1923.5  621.56  2356.1  613.21  2936.2  607.66  2956.2  608.59  3106.2  605.07
  3696.3  598.61  4534.1  596.13  4566.4  596.85  4576.4  595.31  4596.4  596.37
  4632.4   595.6  4836.4  596.34  4906.4  593.12  4936.4  594.25  4976.4  592.76
  4981.3  590.31  4985.4  589.51  5006.6  590.31  5026.5  593.51  5306.8  594.93
  5321.1  595.17  5356.8  599.51  5366.8  597.27  5466.9  597.13    5497  601.21
  5518.8  599.93  5539.2  598.92  5617.1  602.73  6387.9  614.44  6743.4  616.06
#Mann= 6 ,-1 , 0
  1923.5     .05       0  4534.1     .08       0  4632.4      .1       0
  4981.3     .07       0  5006.6      .1       0  5518.8     .05       0
Bank Sta=4981.3,5006.6
XS Rating Curve= 0 ,0
Exp/Cntr=0.3,0.1

Type RM Length L Ch R = 1 ,100073  ,610,610,610
BEGIN DESCRIPTION:
Black Creek 96.0
END DESCRIPTION:
XS GIS Cut Line= 3
      1977531.99     13560615.26       1974125.7     13560662.13
      1972709.56     13561057.82
#Sta/Elev= 30
  1768.5  620.65  2365.5   610.9  2535.6  607.08  2555.6  607.82  2575.6  606.78
  2985.6  601.93  3745.7  595.73  4346.8  594.48  4425.7  595.72  4445.2  594.04
  4455.7  593.96  4465.7   596.6  4543.6  595.55  4705.8  595.55  4775.8  593.38
  4815.8  594.22  4885.8  592.28  4955.8  593.42  4965.8  593.03  4973.1  591.28
  4977.2  590.48  4998.4  591.28  5005.8  592.49  5023.3  592.63    5342  597.22
  5428.8  598.84  5468.1  600.71  5643.1  602.36  6027.2  609.55  6645.5  615.02
#Mann= 7 ,-1 , 0
  1768.5     .05       0  4346.8      .1       0  4445.2     .05       0
  4543.6      .1       0  4973.1     .07       0  4998.4      .1       0
  5023.3     .05       0
Bank Sta=4973.1,4998.4
XS Rating Curve= 0 ,0
Exp/Cntr=0.3,0.1

Type RM Length L Ch R = 1 ,99463   ,1086,1086,1086
BEGIN DESCRIPTION:
Black Creek 95.0
END DESCRIPTION:
XS GIS Cut Line= 3
      1977575.04     13559674.99        1974475.       13560175.
      1972275.04     13560974.99
#Sta/Elev= 30
  1875.9  623.16    2119  621.61  2807.8  606.65  3098.5  602.17  3726.6  595.43
    4202   594.2  4513.1  594.32  4598.5  595.08  4606.8  593.03  4613.2  593.61
  4631.1  592.92  4651.4  595.55  4713.4  594.39  4792.1  592.85  4914.7  594.77
  4920.8   593.1  4975.5  592.02  4982.6  590.27    4983  588.26  4987.2  587.46
  5008.4  588.26  5013.5  591.46    5189  592.28  5228.8  594.14  5835.3  600.81
    6110  605.76  6232.4  605.97  6484.4  610.23  6812.3  612.85  7356.9  623.69
#Mann= 9 ,-1 , 0
  1875.9     .05       0    4202      .1       0  4513.1     .05       0
  4598.5      .1       0  4613.2     .08       0  4713.4      .1       0
    4983     .07       0  5008.4      .1       0    5189     .05       0
Bank Sta=4983,5008.4
XS Rating Curve= 0 ,0
Exp/Cntr=0.3,0.1

Type RM Length L Ch R = 1 ,98377   ,511,511,511
BEGIN DESCRIPTION:
Black Creek 94.0
END DESCRIPTION:
XS GIS Cut Line= 3
      1977405.22     13558865.26        1974775.       13559225.
      1971995.49     13559844.42
#Sta/Elev= 30
  2321.4  623.44  2664.8  619.37    3008  611.57  3159.4   609.4  3603.4  607.24
  3836.5  604.03    4209  595.96  4441.2  592.41  4764.1  591.63  4879.3  592.22
    4966   591.2  4973.6   588.6  4978.7   588.6  4982.5  586.72  4986.7  585.92
    5008  586.72  5017.1  589.85  5109.3  592.35  5474.1   591.2  5509.4  590.98
  5529.4  592.94  5744.5  597.47    6308  599.07  6553.9  598.72  6885.4  600.95
  7640.2  610.21  7714.1  611.44  7732.1  613.03  7757.6  611.79  7823.8   611.8
#Mann= 7 ,-1 , 0
  2321.4     .05       0  4764.1      .1       0  4879.3     .05       0
  4982.5     .07       0    5008     .05       0  5474.1     .05       0
  7640.2      .1       0
Bank Sta=4982.5,5008
XS Rating Curve= 0 ,0
Exp/Cntr=0.3,0.1

Type RM Length L Ch R = 1 ,97866   ,924,924,924
BEGIN DESCRIPTION:
Black Creek 93.0
END DESCRIPTION:
XS GIS Cut Line= 3
      1976884.35      13558497.2        1974525.       13558775.
      1971801.79     13559240.13
#Sta/Elev= 30
    2639  613.96  3282.8  611.79  3777.9  604.55  4263.6  593.41    4330  592.28
  4350.1  597.19  4369.2  597.48  4410.5  590.01  4430.6  589.09  4611.9  589.15
  4642.1  594.27  4662.2  591.61  4762.5  591.22  4793.1  592.24  4823.3  590.41
  4863.6  592.94  4902.7  591.65  4975.6  590.17  4991.8  586.87    4996  586.07
  5017.3  586.87  5024.8  589.88  5034.9  590.22  5102.3  588.91  5267.8  590.56
  5337.8  592.24  6566.8  596.52  6921.9  601.17  7530.6  614.18  7777.3   613.6
#Mann= 7 ,-1 , 0
    2639     .05       0  4263.6      .1       0  4762.5     .05       0
  4902.7      .1       0  4991.8     .07       0  5017.3      .1       0
  5267.8     .05       0
Bank Sta=4991.8,5017.3
XS Rating Curve= 0 ,0
Exp/Cntr=0.3,0.1
