--- Horse Creek.prj (project) ---

Proj Title=Horse Creek Base Level Engineering
Current Plan=p01
Default Exp/Contr=0.3,0.1
English Units
Geom File=g01
Flow File=f01
Plan File=p01
Y Axis Title=Elevation
X Axis Title(PF)=Main Channel Distance
X Axis Title(XS)=Station
BEGIN DESCRIPTION:
Horse Creek
END DESCRIPTION:
DSS Export Rating Curves= 0
DSS Export Rating Curve Sorted= 0
DSS Export Volume Flow Curves= 0
DXF OffsetX= 0
DXF OffsetY= 0
DXF ScaleX= 1
DXF ScaleY= 10

--- Horse Creek.p01 (plan) ---

Plan Title=Multiple Run
Short Identifier=Multiple
Geom File=g01
Flow File=f01
Subcritical Flow
K Sum by GR= 0
Std Step Tol= 0.01
Critical Tol= 0.01
Num of Std Step Trials= 20
Max Error Tol= 0.3
Flow Tol Ratio= 0.001
Split Flow NTrial= 30
Split Flow Tol= 0.02
Split Flow Ratio= 0.02
Log Output Level= 0
Friction Slope Method= 1
Unsteady Friction Slope Method= 2
Unsteady Bridges Friction Slope Method= 1
Parabolic Critical Depth
Global Vel Dist=  1 , 1 , 1
Global Log Level= 0
CheckData=True
Encroach Param= -1, 0, 0, 0
BEGIN DESCRIPTION:
Multiple Run
END DESCRIPTION:

--- Horse Creek.f01 (steady flow) ---

Flow Title=Multiple
Program Version=5.05
Number of Profiles= 7
Profile Names=10-year,25-year,50-year,1pct_min,100-year,1pct_plu,500-year
River Rch & RM=Horse Creek,Reach-1         ,35557
     100     134     161      98     195     390     290
River Rch & RM=Horse Creek,Reach-1         ,28502
     708    1026    1300     816    1629    3249    2583
River Rch & RM=Horse Creek,Reach-1         ,23194
    1539    2299    2970    1894    3780    7541    6170
River Rch & RM=Horse Creek,Reach-1         ,21439
    1446    2156    2781    1773    3538    7059    5777
River Rch & RM=Horse Creek,Reach-1         ,19468
    1339    1990    2564    1635    3262    6509    5342
River Rch & RM=Horse Creek,Reach-1         ,17636
    1339    1990    2564    1635    3262    6509    5342
River Rch & RM=Horse Creek,Reach-1         ,10196
    1304    1931    2481    1578    3149    6283    5132
Boundary for River Rch & Prof#=Horse Creek,Reach-1         , 1
Up Type= 0
Dn Type= 3
Dn Slope=0.0021
Boundary for River Rch & Prof#=Horse Creek,Reach-1         , 2
Up Type= 0
Dn Type= 3
Dn Slope=0.0021
Boundary for River Rch & Prof#=Horse Creek,Reach-1         , 3
Up Type= 0
Dn Type= 3
Dn Slope=0.0021
Boundary for River Rch & Prof#=Horse Creek,Reach-1         , 4
Up Type= 0
Dn Type= 3
Dn Slope=0.0021
Boundary for River Rch & Prof#=Horse Creek,Reach-1         , 5
Up Type= 0
Dn Type= 3
Dn Slope=0.0021
Boundary for River Rch & Prof#=Horse Creek,Reach-1         , 6
Up Type= 0
Dn Type= 3
Dn Slope=0.0021
Boundary for River Rch & Prof#=Horse Creek,Reach-1         , 7
Up Type= 0
Dn Type= 3
Dn Slope=0.0021
DSS Import GetInterval= 0
DSS Import GetPeak= 0
DSS Import FillOption= 0

--- Horse Creek.g01 (geometry) ---

Geom Title=Existing Conditions

River Reach=Horse Creek,Reach-1
Reach XY= 30
      1956185.80     13542709.54      1957017.26     13544193.67
      1957900.80     13544224.54      1959250.80     13545544.54
      1959520.80     13545474.54      1960070.80     13546364.54
      1962170.80     13545474.54      1962860.80     13544704.54
      1963860.80     13544634.54      1963970.80     13544104.54
      1964330.80     13544174.54      1964740.80     13543644.54
      1964610.80     13542944.54      1965240.80     13542864.54
      1965130.80     13542374.54      1966200.80     13542154.54
      1967020.80     13540994.54      1967108.47     13540300.72
      1968094.58     13539750.03      1968630.80     13539804.54
      1969030.80     13539124.54      1969960.80     13539094.54
      1970320.80     13538664.54      1971990.80     13539334.54
      1972090.80     13539624.54      1972810.80     13539314.54
      1973910.80     13539824.54      1974660.80     13539434.54
      1974840.80     13539614.54      1975500.80     13538814.54

Type RM Length L Ch R = 1,35557,348,348,348
BEGIN DESCRIPTION:
Horse Creek 36.0
END DESCRIPTION:
XS GIS Cut Line= 3
      1955851.20     13542905.51      1956456.64     13542829.55
      1956610.34     13542716.99
#Sta/Elev= 30
  4677.9  707.95  4752.3  703.86  4800.0  699.48  4805.1  699.55  4822.8  697.41
  4880.5  693.01  4933.7  690.15  4961.0  689.03  4966.1  689.42  4982.1  688.84
  4982.3  688.34  4985.8  688.34  4986.1  688.84  5024.4  688.95  5046.5  689.69
  5094.9  690.22  5135.3  691.25  5195.7  691.81  5246.1  693.16  5282.9  693.20
  5298.3  693.59  5304.4  694.16  5319.1  694.17  5325.3  694.86  5354.6  695.52
  5360.8  696.54  5369.3  696.42  5375.5  697.14  5419.5  698.22  5478.6  700.69
#Mann=3,-1,0
  4677.9     0.1       0  4982.1    0.07       0  4986.1     0.1       0
Bank Sta=4982.1,4986.1
Exp/Cntr=0.3,0.1

Type RM Length L Ch R = 1,35209,341,341,341
BEGIN DESCRIPTION:
Mapping XS 868b6979
END DESCRIPTION:
XS GIS Cut Line= 4
      1955954.32     13543153.30      1956131.43     13543200.19
      1956475.18     13543116.85      1956615.80     13542931.98
#Sta/Elev= 30
  4688.4  701.39  4714.8  699.65  4755.0  696.02  4782.2  693.03  4790.1  691.54
  4802.9  690.41  4865.0  686.82  4870.5  686.08  4913.1  685.07  4960.0  684.77
  4978.2  684.19  4999.8  682.21  5000.1  681.71  5003.6  681.71  5003.8  682.21
  5019.3  683.78  5043.6  683.45  5050.2  682.75  5085.4  683.69  5111.9  683.09
  5153.1  683.43  5169.0  682.68  5194.3  683.15  5210.8  682.85  5312.6  684.65
  5340.7  684.31  5377.0  685.69  5404.1  686.02  5447.8  688.61  5457.6  688.71
#Mann=3,-1,0
  4688.4     0.1       0  4999.8    0.07       0  5003.8     0.1       0
Bank Sta=4999.8,5003.8
Exp/Cntr=0.3,0.1

Type RM Length L Ch R = 1,34868,231,231,231
BEGIN DESCRIPTION:
Mapping XS cbc02a52
END DESCRIPTION:
XS GIS Cut Line= 4
      1956058.48     13543374.66      1956308.52     13543398.10
      1956649.66     13543192.38      1956766.86     13542971.00
#Sta/Elev= 30
  4470.1  686.47  4476.7  685.86  4534.7  683.99  4567.0  683.28  4627.3  681.06
  4697.6  680.17  4735.8  678.82  4792.0  678.43  4792.3  677.93  4795.8  677.93
  4796.0  678.43  4801.3  678.60  4852.3  678.72  4895.0  680.03  4910.5  679.11
  4939.0  679.85  4968.7  678.66  4974.6  679.32  4990.1  679.63  5085.2  679.16
  5106.6  679.71  5119.6  679.52  5203.7  681.52  5231.3  681.70  5275.3  683.19
  5286.0  683.08  5320.3  685.48  5335.7  685.79  5352.0  686.97  5370.1  687.50
#Mann=5,-1,0
  4470.1     0.1       0  4534.7    0.05       0  4792.0    0.07       0
  4796.0    0.05       0  4801.3     0.1       0
Bank Sta=4792,4796
Exp/Cntr=0.3,0.1

Type RM Length L Ch R = 1,34637,63,63,63
BEGIN DESCRIPTION:
Mapping XS 975f1454
END DESCRIPTION:
XS GIS Cut Line= 5
      1956089.76     13543411.13      1956404.87     13543418.94
      1956733.77     13543408.97      1956995.93     13543382.22
      1957031.82     13543373.55
#Sta/Elev= 30
  4376.8  684.86  4382.0  684.36  4408.8  683.66  4432.1  682.62  4472.1  681.69
  4482.1  681.05  4522.1  680.29  4542.1  680.58  4632.1  678.27  4662.1  677.16
  4702.1  677.62  4732.2  676.49  4822.2  676.78  4872.2  675.07  4922.2  674.78
  4970.3  673.06  4970.5  672.56  4974.0  672.56  4974.3  673.06  4987.2  673.86
  5042.4  674.16  5052.4  673.74  5098.2  674.40  5173.1  676.78  5197.4  676.74
  5208.1  676.77  5213.3  676.42  5296.9  677.00  5306.5  676.63  5321.5  676.64
#Mann=8,-1,0
  4376.8     0.1       0  4408.8    0.05       0  4970.3    0.04       0
  4974.3    0.05       0  5098.2    0.08       0  5197.4    0.05       0
  5296.9    0.08       0  5306.5     0.1       0
Bank Sta=4970.3,4974.3
Exp/Cntr=0.3,0.1

Type RM Length L Ch R = 1,34574,305,305,305
BEGIN DESCRIPTION:
Mapping XS 16589032
END DESCRIPTION:
XS GIS Cut Line= 3
      1956193.91     13543517.90      1956739.97     13543469.24
      1957045.44     13543436.90
#Sta/Elev= 30
  4463.6  680.47  4484.8  680.47  4504.9  679.25  4605.2  678.01  4705.6  675.39
  4725.7  675.84  4774.4  674.64  4779.4  675.13  4806.0  675.32  4826.1  674.37
  4886.0  673.53  4891.0  674.05  4926.5  673.60  4946.6  673.71  4956.6  673.05
  4966.7  673.76  4984.6  672.69  5016.9  672.42  5037.0  672.75  5075.2  672.00
  5075.5  671.50  5079.0  671.50  5079.2  672.00  5080.9  672.09  5137.6  675.03
  5180.1  676.09  5193.7  676.16  5198.7  675.44  5279.3  675.16  5319.0  674.59
#Mann=7,-1,0
  4463.6     0.1       0  4984.6    0.05       0  5075.2    0.04       0
  5079.2    0.05       0  5080.9    0.08       0  5180.1    0.05       0
  5279.3    0.08       0
Bank Sta=5075.2,5079.2
Exp/Cntr=0.3,0.1

Type RM Length L Ch R = 1,34269,212,212,212
BEGIN DESCRIPTION:
Mapping XS 957b21b0
END DESCRIPTION:
XS GIS Cut Line= 4
      1956225.21     13543653.32      1956550.70     13543728.83
      1956742.83     13543701.33      1956892.47     13543469.08
#Sta/Elev= 30
  4517.8  677.94  4588.0  676.20  4620.2  676.11  4683.5  674.67  4726.2  674.23
  4753.7  674.43  4835.8  672.76  4846.1  672.87  4937.1  671.35  4967.4  670.39
  5026.0  669.40  5026.3  668.90  5029.8  668.90  5030.0  669.40  5095.7  670.11
  5153.1  669.62  5160.6  669.90  5168.3  670.83  5174.2  670.71  5189.4  671.56
  5204.6  670.50  5219.8  671.02  5232.0  671.94  5240.9  671.91  5246.9  672.47
  5255.8  672.56  5277.2  674.04  5283.2  673.94  5319.3  675.20  5322.3  675.46
#Mann=4,-1,0
  4517.8     0.1       0  5026.0    0.07       0  5030.0     0.1       0
  5319.3    0.08       0
Bank Sta=5026,5030
Exp/Cntr=0.3,0.1

Type RM Length L Ch R = 1,34057,69,69,69
BEGIN DESCRIPTION:
Mapping XS b6ec9747
END DESCRIPTION:
XS GIS Cut Line= 4
      1956305.93     13543866.86      1956602.79     13543913.73
      1956797.52     13543878.41      1956886.56     13543512.43
#Sta/Elev= 30
  4511.4  674.23  4663.6  671.17  4753.4  670.65  4831.1  668.80  4865.0  668.57
  4915.8  667.15  5031.9  665.95  5032.2  665.45  5035.7  665.45  5035.9  665.95
  5044.2  666.35  5095.7  666.16  5102.9  666.76  5108.0  666.45  5116.3  667.41
  5126.6  666.93  5144.6  668.23  5157.4  668.50  5191.5  668.42  5228.1  669.08
  5233.2  668.61  5275.0  668.90  5280.9  669.57  5301.5  669.78  5311.6  670.67
  5316.7  670.58  5332.4  672.38  5353.0  672.69  5358.4  673.27  5386.5  674.14
#Mann=3,-1,0
  4511.4     0.1       0  5031.9    0.07       0  5035.9     0.1       0
Bank Sta=5031.9,5035.9
Exp/Cntr=0.3,0.1

Type RM Length L Ch R = 1,33988,337,337,337
BEGIN DESCRIPTION:
Mapping XS 16d5d0cf
END DESCRIPTION:
XS GIS Cut Line= 4
      1956326.71     13544166.34      1956644.45     13544137.69
      1956826.16     13544064.61      1956907.39     13543533.27
#Sta/Elev= 30
  4324.3  681.01  4372.8  678.90  4443.1  673.74  4513.4  670.29  4573.6  667.92
  4654.7  666.62  4695.8  663.43  4696.1  662.93  4699.6  662.93  4699.8  663.43
  4708.6  665.09  4730.2  665.62  4784.0  664.44  4799.1  664.54  4835.9  663.46
  4990.5  664.99  5010.8  664.01  5051.2  665.26  5091.7  665.49  5122.0  666.50
  5152.4  666.70  5182.7  668.01  5203.0  667.74  5265.2  668.26  5273.8  669.20
  5283.9  669.06  5304.1  670.37  5328.6  670.51  5344.6  672.02  5376.7  673.99
#Mann=3,-1,0
  4324.3     0.1       0  4695.8    0.07       0  4699.8     0.1       0
Bank Sta=4695.8,4699.8
Exp/Cntr=0.3,0.1

Type RM Length L Ch R = 1,33651,189,189,189
BEGIN DESCRIPTION:
Mapping XS f3f06e43
END DESCRIPTION:
XS GIS Cut Line= 4
      1956597.62     13544510.06      1956868.41     13544356.44
      1957071.54     13544043.94      1957128.83     13543734.04
#Sta/Elev= 30
  4414.3  673.84  4459.0  671.86  4526.3  670.48  4561.4  668.67  4571.5  668.67
  4577.3  667.88  4593.2  668.01  4598.9  667.11  4614.8  667.22  4620.5  666.39
  4636.4  666.40  4642.2  665.82  4664.2  665.24  4673.9  665.02  4687.2  665.72
  4722.0  664.46  4846.6  661.92  4897.0  659.74  4948.4  659.96  4988.6  659.32
  4988.8  658.82  4992.3  658.82  4992.6  659.32  5078.2  659.58  5085.2  659.70
  5093.3  660.74  5107.4  660.97  5149.1  661.00  5312.9  663.37  5413.5  666.57
#Mann=3,-1,0
  4414.3     0.1       0  4988.6    0.07       0  4992.6     0.1       0
Bank Sta=4988.6,4992.6
Exp/Cntr=0.3,0.1

Type RM Length L Ch R = 1,33462,96,96,96
BEGIN DESCRIPTION:
Mapping XS e46a0cd1
END DESCRIPTION:
XS GIS Cut Line= 4
      1956831.93     13544715.84      1957097.58     13544366.85
      1957209.56     13543913.73      1957152.26     13543723.62
#Sta/Elev= 30
  4393.0  673.74  4459.5  670.86  4482.0  670.64  4567.6  668.01  4632.0  665.48
  4652.8  665.12  4659.1  665.78  4673.7  664.45  4738.1  662.63  4752.6  662.79
  4796.2  661.56  4802.5  661.82  4808.8  661.30  4823.4  661.36  4915.9  659.52
  5099.2  659.68  5101.5  659.66  5176.9  659.47  5213.1  660.07  5222.9  659.37
  5223.2  658.87  5226.7  658.87  5226.9  659.37  5254.6  659.52  5276.4  661.00
  5332.5  661.98  5338.8  662.54  5403.7  663.34  5464.1  666.19  5496.9  667.24
#Mann=5,-1,0
  4393.0     0.1       0  5099.2    0.05       0  5101.5     0.1       0
  5222.9    0.07       0  5226.9     0.1       0
Bank Sta=5222.9,5226.9
Exp/Cntr=0.3,0.1

Type RM Length L Ch R = 1,33366,37,37,37
BEGIN DESCRIPTION:
Mapping XS 47dfc213
END DESCRIPTION:
XS GIS Cut Line= 4
      1956950.56     13544845.63      1957172.79     13544467.14
      1957311.68     13543880.34      1957285.08     13543515.33
#Sta/Elev= 30
  4293.5  674.74  4398.6  670.28  4503.0  667.33  4546.4  665.36  4552.1  665.67
  4560.9  665.45  4605.0  663.51  4618.9  663.26  4626.4  663.55  4669.4  661.65
  4736.1  661.43  4767.1  660.25  4804.3  659.73  5018.1  659.81  5102.6  659.41
  5102.8  658.91  5106.3  658.91  5106.6  659.41  5130.7  659.64  5269.0  659.79
  5320.4  661.03  5340.8  661.01  5411.0  662.46  5431.0  663.71  5461.1  664.55
  5481.1  664.54  5591.4  667.45  5611.5  667.42  5651.6  668.66  5701.4  669.32
#Mann=5,-1,0
  4293.5     0.1       0  5018.1    0.05       0  5102.6    0.07       0
  5106.6    0.05       0  5130.7     0.1       0
Bank Sta=5102.6,5106.6
Exp/Cntr=0.3,0.1

Type RM Length L Ch R = 1,33329,45,45,45
BEGIN DESCRIPTION:
Horse Creek 32.0
END DESCRIPTION:
XS GIS Cut Line= 4
      1957004.84     13544842.11      1957204.47     13544484.07
      1957371.58     13543789.62      1957342.37     13543502.31
#Sta/Elev= 30
  4305.7  673.18  4523.7  665.13  4683.9  661.24  4684.2  660.74  4687.9  661.24
  4701.9  661.90  4712.2  663.79  4745.5  665.51  4807.3  665.27  4823.7  664.29
  4828.9  665.72  4865.7  664.56  4870.8  665.72  4907.6  664.92  4920.4  666.01
  4949.5  664.73  4954.7  665.98  4991.5  664.56  4996.6  665.69  5038.6  666.34
  5080.5  664.50  5085.7  665.62  5122.5  664.56  5127.6  665.55  5187.8  665.20
  5206.3  664.13  5352.4  664.92  5403.8  662.45  5426.3  662.52  5718.7  668.64
#Mann=3,-1,0
  4305.7     0.1       0  4683.9    0.07       0  4687.9     0.1       0
Bank Sta=4683.9,4687.9
Exp/Cntr=0.3,0.1

Type RM Length L Ch R = 1,33284,258,258,258
BEGIN DESCRIPTION:
Mapping XS 1d5b6e26
END DESCRIPTION:
XS GIS Cut Line= 5
      1957030.45     13544838.63      1957249.18     13544487.97
      1957367.24     13543991.45      1957422.79     13543751.86
      1957397.06     13543504.89
#Sta/Elev= 30
  4299.6  672.41  4487.1  665.42  4654.7  660.89  4681.8  660.67  4704.6  661.72
  4711.7  660.69  4718.8  661.18  4726.2  660.00  4736.5  659.49  4845.3  657.88
  4921.5  655.87  4981.2  653.29  4981.4  652.79  4984.9  652.79  4985.2  653.29
  5014.0  654.42  5019.1  653.42  5061.3  655.93  5066.4  654.76  5103.5  655.28
  5108.6  654.22  5137.4  654.65  5187.8  656.84  5192.9  656.37  5283.0  658.38
  5383.8  661.34  5458.8  661.96  5536.4  663.86  5576.6  664.16  5717.5  667.66
#Mann=3,-1,0
  4299.6     0.1       0  4981.2    0.07       0  4985.2     0.1       0
Bank Sta=4981.2,4985.2
Exp/Cntr=0.3,0.1

Type RM Length L Ch R = 1,33026,276,276,276
BEGIN DESCRIPTION:
Horse Creek 31.0
END DESCRIPTION:
XS GIS Cut Line= 3
      1957269.46     13544705.38      1957590.76     13544210.63
      1957649.62     13543609.53
#Sta/Elev= 30
  4460.2  664.18  4572.6  660.34  4593.7  659.78  4602.9  660.13  4608.9  659.29
  4746.8  655.82  4769.0  654.78  4790.1  655.04  4847.5  653.66  4898.9  653.81
  4935.1  653.01  4977.3  651.47  4992.4  648.65  4996.4  648.39  4996.7  647.89
  5000.2  647.89  5000.4  648.39  5013.6  648.93  5021.1  650.71  5028.7  650.99
  5049.4  650.40  5085.9  651.62  5176.4  651.36  5226.6  653.65  5346.2  656.36
  5477.8  657.87  5518.0  659.28  5588.3  660.69  5598.4  660.31  5654.1  661.34
#Mann=3,-1,0
  4460.2     0.1       0  4996.4    0.07       0  5000.4     0.1       0
Bank Sta=4996.4,5000.4
Exp/Cntr=0.3,0.1

Type RM Length L Ch R = 1,32750,30,30,30
BEGIN DESCRIPTION:
Mapping XS 6594c7a3
END DESCRIPTION:
XS GIS Cut Line= 6
      1957353.60     13544725.43      1957652.18     13544407.75
      1957719.89     13544308.79      1957808.43     13544235.87
      1957853.57     13544138.65      1958093.11     13543709.90
#Sta/Elev= 30
  4295.7  663.36  4360.7  661.46  4395.9  659.72  4749.3  649.25  4794.1  648.32
  4800.1  649.07  4858.2  647.45  4865.0  648.09  4871.5  647.56  4879.4  648.96
  4900.2  649.87  4928.9  646.92  4961.0  646.63  4961.3  646.13  4964.8  646.13
  4965.0  646.63  4971.4  647.44  4988.8  646.70  4994.3  647.58  5000.3  646.90
  5055.4  647.07  5072.7  648.66  5100.6  649.79  5171.8  650.92  5209.5  652.28
  5252.9  652.05  5268.9  652.89  5296.3  652.77  5350.0  654.10  5564.6  656.22
#Mann=3,-1,0
  4295.7     0.1       0  4961.0    0.07       0  4965.0     0.1       0
Bank Sta=4961,4965
Exp/Cntr=0.3,0.1

Type RM Length L Ch R = 1,32720,63,63,63
BEGIN DESCRIPTION:
Mapping XS 5ce83773
END DESCRIPTION:
XS GIS Cut Line= 6
      1957346.63     13544741.08      1957674.75     13544421.64
      1957702.53     13544362.61      1957839.68     13544244.55
      1957862.25     13544183.79      1958148.72     13543695.92
#Sta/Elev= 30
  4261.2  664.07  4377.5  659.72  4681.5  650.87  4726.2  650.95  4777.3  650.10
  4919.6  650.99  4925.7  649.98  4934.2  651.02  4940.4  650.10  4947.6  650.66
  4955.1  650.14  4961.1  651.19  4965.7  651.19  4968.6  650.21  4975.9  651.49
  5024.0  650.89  5032.7  651.53  5075.5  650.91  5089.1  649.11  5096.7  649.06
  5097.0  648.56  5100.5  648.56  5100.7  649.06  5222.0  651.96  5249.5  651.63
  5302.1  652.92  5345.1  653.01  5360.7  653.95  5462.3  654.25  5596.3  656.33
#Mann=3,-1,0
  4261.2     0.1       0  5096.7    0.07       0  5100.7     0.1       0
Bank Sta=5096.7,5100.7
Exp/Cntr=0.3,0.1

Type RM Length L Ch R = 1,32657,104,104,104
BEGIN DESCRIPTION:
Mapping XS 4bb3c8d3
END DESCRIPTION:
XS GIS Cut Line= 3
      1957386.76     13544746.23      1957998.75     13544144.66
      1958323.80     13543749.40
#Sta/Elev= 30
  4267.6  662.96  4288.5  661.65  4337.9  660.56  4387.5  658.00  4451.1  657.07
  4472.3  655.82  4507.6  655.39  4514.8  654.55  4585.5  652.60  4592.5  652.91
  4613.8  651.82  4663.2  651.25  4790.5  648.04  4931.9  647.34  4960.2  646.44
  4995.5  643.60  5007.7  643.32  5007.9  642.82  5011.4  642.82  5011.7  643.32
  5108.7  648.35  5158.4  649.48  5222.3  649.53  5228.9  650.45  5271.8  650.80
  5413.9  651.00  5436.0  651.46  5442.6  652.19  5449.0  651.63  5637.5  653.08
#Mann=3,-1,0
  4267.6     0.1       0  5007.7    0.07       0  5011.7     0.1       0
Bank Sta=5007.7,5011.7
Exp/Cntr=0.3,0.1

Type RM Length L Ch R = 1,32553,670,670,670
BEGIN DESCRIPTION:
Horse Creek 30.0
END DESCRIPTION:
XS GIS Cut Line= 3
      1957470.12     13544811.30      1957954.47     13544326.95
      1958444.07     13543821.73
#Sta/Elev= 30
  4294.7  659.42  4422.8  654.23  4429.9  655.04  4437.0  654.05  4472.3  654.60
  4507.7  653.34  4550.1  654.40  4663.2  653.28  4762.2  648.73  4854.1  646.22
  4882.4  643.31  4896.6  642.72  4929.9  642.25  4930.2  641.75  4933.9  642.25
  4939.0  643.75  4953.1  644.11  4974.4  642.97  4977.5  644.33  4995.7  643.46
  5002.6  642.25  5016.8  642.52  5024.0  644.24  5045.1  645.46  5172.4  647.74
  5278.4  647.40  5441.2  649.01  5490.6  648.61  5518.9  649.65  5683.2  649.90
#Mann=3,-1,0
  4294.7     0.1       0  4929.9    0.07       0  4933.9     0.1       0
Bank Sta=4929.9,4933.9
Exp/Cntr=0.3,0.1

Type RM Length L Ch R = 1,31883,442,442,442
BEGIN DESCRIPTION:
Horse Creek 29.0
END DESCRIPTION:
XS GIS Cut Line= 4
      1957613.29     13545076.96      1958126.35     13544951.95
      1958550.83     13544639.45      1958592.10     13544445.47
#Sta/Elev= 30
  4155.9  656.62  4226.1  653.15  4250.3  652.56  4291.5  649.57  4415.0  645.97
  4439.7  647.01  4476.3  646.71  4528.3  647.67  4548.8  647.05  4564.8  645.09
  4589.9  647.98  4611.7  648.49  4653.4  648.09  4838.3  641.35  4923.9  639.25
  4938.6  637.43  4944.8  638.11  4953.2  637.84  4974.1  635.64  4980.3  634.40
  4986.7  634.23  4986.9  633.73  4990.4  633.73  4990.7  634.23  5017.6  634.26
  5030.4  636.38  5053.5  637.12  5124.5  636.76  5338.3  639.32  5409.4  639.56
#Mann=3,-1,0
  4155.9     0.1       0  4986.7    0.07       0  4990.7     0.1       0
Bank Sta=4986.7,4990.7
Exp/Cntr=0.3,0.1

Type RM Length L Ch R = 1,31441,452,452,452
BEGIN DESCRIPTION:
Horse Creek 28.0
END DESCRIPTION:
XS GIS Cut Line= 3
      1958075.00     13545625.00      1958675.00     13545025.00
      1958833.80     13544699.06
#Sta/Elev= 30
  4149.9  650.37  4234.8  644.53  4319.6  641.58  4545.9  637.19  4560.0  636.64
  4574.2  635.34  4588.3  635.12  4616.6  635.98  4786.3  634.47  4800.4  633.88
  4956.0  633.30  4970.1  632.96  4984.3  631.10  4992.9  629.03  4993.1  628.53
  4996.6  628.53  4996.9  629.03  5001.2  629.03  5020.7  632.34  5029.5  632.70
  5035.0  631.81  5052.0  631.77  5065.2  631.13  5080.1  631.26  5109.7  632.75
  5125.2  632.78  5176.4  635.17  5266.0  636.93  5328.0  637.13  5361.0  636.45
#Mann=3,-1,0
  4149.9     0.1       0  4992.9    0.07       0  4996.9     0.1       0
Bank Sta=4992.9,4996.9
Exp/Cntr=0.3,0.1

Type RM Length L Ch R = 1,30989,351,351,351
BEGIN DESCRIPTION:
Horse Creek 27.0
END DESCRIPTION:
XS GIS Cut Line= 3
      1958374.97     13545875.03      1958975.00     13545275.00
      1959173.23     13544936.32
#Sta/Elev= 30
  4139.3  641.89  4167.6  640.22  4464.6  632.82  4478.8  631.97  4507.0  632.16
  4535.3  631.18  4775.7  629.68  4832.3  628.51  4846.5  629.36  4931.3  628.41
  4959.6  629.01  4990.8  627.43  4999.5  625.29  4999.8  624.79  5003.3  624.79
  5003.5  625.29  5011.1  626.63  5023.0  625.59  5038.7  626.43  5045.8  625.97
  5060.2  628.61  5075.9  630.06  5171.7  635.39  5177.5  634.96  5214.7  635.71
  5236.2  635.50  5251.9  636.18  5279.1  635.61  5332.0  635.99  5380.3  635.47
#Mann=3,-1,0
  4139.3     0.1       0  4999.5    0.07       0  5003.5     0.1       0
Bank Sta=4999.5,5003.5
Exp/Cntr=0.3,0.1

Type RM Length L Ch R = 1,30638,710,710,710
BEGIN DESCRIPTION:
Horse Creek 26.0
END DESCRIPTION:
XS GIS Cut Line= 3
      1958473.60     13546048.72      1959227.04     13545461.93
      1959660.53     13545090.87
#Sta/Elev= 30
  4072.7  641.30  4212.3  637.43  4411.4  630.74  4432.2  630.78  4703.6  625.47
  4738.9  626.18  4759.7  625.82  4782.3  624.02  4788.7  624.36  4796.8  623.87
  4809.6  625.03  4838.4  625.88  4896.3  625.62  4987.7  623.77  5002.2  622.62
  5008.3  620.89  5008.6  620.39  5012.1  620.39  5012.3  620.89  5016.7  623.52
  5023.2  624.24  5080.5  625.15  5102.5  624.86  5123.3  625.48  5208.9  625.89
  5264.9  627.62  5406.7  629.93  5428.5  629.68  5463.6  630.44  5598.3  630.21
#Mann=3,-1,0
  4072.7     0.1       0  5008.3    0.07       0  5012.3     0.1       0
Bank Sta=5008.3,5012.3
Exp/Cntr=0.3,0.1

Type RM Length L Ch R = 1,29928,456,456,456
BEGIN DESCRIPTION:
Horse Creek 25.0
END DESCRIPTION:
XS GIS Cut Line= 3
      1958529.15     13546152.90      1959625.00     13545675.00
      1960015.23     13545444.58
#Sta/Elev= 30
  3770.7  640.30  3879.4  637.78  3902.8  636.76  4054.2  632.71  4115.3  629.89
  4129.9  630.20  4229.0  627.74  4497.1  622.65  4526.4  622.47  4573.2  620.01
  4631.0  620.63  4671.7  620.52  4677.8  620.10  4777.0  620.79  4889.9  620.42
  4928.4  619.59  4979.8  620.03  4989.4  619.68  4999.3  616.93  4999.5  616.43
  5003.0  616.43  5003.3  616.93  5016.9  617.17  5024.3  619.27  5032.6  619.73
  5163.6  624.46  5214.0  627.29  5331.1  631.06  5346.7  630.95  5419.4  632.58
#Mann=3,-1,0
  3770.7     0.1       0  4999.3    0.07       0  5003.3     0.1       0
Bank Sta=4999.3,5003.3
Exp/Cntr=0.3,0.1

Type RM Length L Ch R = 1,29472,486,486,486
BEGIN DESCRIPTION:
Horse Creek 24.0
END DESCRIPTION:
XS GIS Cut Line= 3
      1958664.50     13546413.34      1959612.46     13546076.52
      1960199.23     13545465.44
#Sta/Elev= 30
  3880.6  635.09  4160.9  629.25  4222.6  627.27  4242.0  625.96  4263.2  626.73
  4475.4  622.54  4756.7  618.11  4910.7  617.33  4924.9  617.05  4939.0  615.53
  4946.0  615.44  4960.1  615.47  4967.3  616.66  4988.4  616.81  4995.6  616.23
  5000.6  612.88  5000.8  612.38  5004.3  612.38  5004.6  612.88  5030.9  616.13
  5186.5  617.68  5306.7  621.42  5483.7  628.44  5526.1  629.31  5547.2  628.97
  5589.7  631.29  5596.6  630.93  5618.0  631.98  5681.5  633.23  5733.8  633.62
#Mann=3,-1,0
  3880.6     0.1       0  5000.6    0.07       0  5004.6     0.1       0
Bank Sta=5000.6,5004.6
Exp/Cntr=0.3,0.1

Type RM Length L Ch R = 1,28986,484,484,484
BEGIN DESCRIPTION:
Horse Creek 23.0
END DESCRIPTION:
XS GIS Cut Line= 4
      1958543.05     13546632.07      1959578.22     13546632.49
      1960177.13     13546126.86      1960388.83     13545439.71
#Sta/Elev= 30
  3496.1  635.90  3598.1  631.86  3768.1  626.84  4138.1  619.50  4527.2  614.35
  4577.2  615.02  4875.0  613.01  4973.9  613.26  4981.6  612.99  4986.2  609.29
  4986.4  608.79  4990.2  609.29  5010.2  611.67  5016.8  613.31  5031.0  611.45
  5037.6  612.49  5045.3  611.34  5051.9  613.18  5059.6  612.09  5066.2  613.23
  5073.9  611.82  5094.8  613.18  5286.1  612.37  5318.7  611.45  5497.4  614.07
  5736.6  622.92  5834.6  628.01  5932.7  634.66  5937.9  633.98  6034.1  634.78
#Mann=3,-1,0
  3496.1     0.1       0  4986.2    0.07       0  4990.2     0.1       0
Bank Sta=4986.2,4990.2
Exp/Cntr=0.3,0.1

Type RM Length L Ch R = 1,28502,260,260,260
BEGIN DESCRIPTION:
Horse Creek 22.0
END DESCRIPTION:
XS GIS Cut Line= 3
      1960693.20     13547444.59      1960315.59     13546272.70
      1960342.03     13545718.36
#Sta/Elev= 30
  3722.4  619.52  3767.3  619.02  3848.0  616.60  4023.8  613.93  4278.8  611.13
  4384.7  611.29  4611.5  611.48  4784.8  610.44  4841.2  610.33  4873.2  609.00
  4930.2  609.36  4937.3  608.61  4942.6  610.21  4971.3  610.70  4987.3  608.47
  4987.8  607.97  4995.5  608.47  5001.4  608.50  5011.4  610.58  5021.4  611.00
  5071.5  611.18  5091.5  610.49  5161.6  611.22  5311.7  614.29  5371.8  616.72
  5391.8  618.36  5411.8  618.18  5451.9  620.46  5466.5  620.52  5508.6  623.54
#Mann=5,-1,0
  3722.4     0.1       0  4384.7    0.05       0  4784.8     0.1       0
  4987.3    0.07       0  4995.5     0.1       0
Bank Sta=4987.3,4995.5
Exp/Cntr=0.3,0.1

Type RM Length L Ch R = 1,28242,47,47,47
BEGIN DESCRIPTION:
Mapping XS 0e0edb58
END DESCRIPTION:
XS GIS Cut Line= 4
      1960982.26     13547501.88      1960596.84     13546454.99
      1960497.88     13546012.28      1960404.48     13545789.16
#Sta/Elev= 30
  3665.2  619.10  3693.8  618.75  3699.9  618.17  3755.5  618.00  3768.4  618.63
  3786.0  617.53  3853.7  616.44  4024.3  615.12  4088.1  613.68  4322.6  612.21
  4363.4  611.32  4525.0  609.72  4773.5  610.65  4904.0  609.27  4934.5  608.41
  4971.4  608.31  4971.9  607.81  4979.1  607.81  4979.6  608.31  5036.6  608.39
  5047.2  610.02  5057.4  609.18  5077.9  610.32  5170.1  609.17  5264.0  611.23
  5274.8  610.82  5404.9  614.74  5415.8  615.86  5457.9  617.24  5476.3  618.45
#Mann=5,-1,0
  3665.2     0.1       0  4363.4    0.05       0  4904.0     0.1       0
  4971.4    0.07       0  4979.6     0.1       0
Bank Sta=4971.4,4979.6
Exp/Cntr=0.3,0.1

Type RM Length L Ch R = 1,28195,38,38,38
BEGIN DESCRIPTION:
Mapping XS 4bdde867
END DESCRIPTION:
XS GIS Cut Line= 4
      1960995.28     13547507.10      1960648.92     13546449.78
      1960492.67     13545876.86      1960422.37     13545744.07
#Sta/Elev= 30
  3637.6  619.10  3973.5  614.64  3978.8  615.20  4069.1  613.72  4092.3  613.62
  4100.9  614.18  4123.9  613.24  4155.4  613.66  4208.0  612.59  4331.2  611.95
  4429.9  610.24  4530.2  609.40  4530.7  608.90  4537.9  608.90  4538.4  609.40
  4629.0  610.38  4702.6  610.01  4716.5  610.45  4723.7  611.49  4743.1  612.58
  4782.6  613.87  4890.6  613.12  5015.8  611.91  5159.2  612.55  5164.4  611.87
  5221.6  612.79  5304.5  611.85  5372.8  614.40  5455.1  619.29  5494.3  620.98
#Mann=5,-1,0
  3637.6     0.1       0  4331.2    0.05       0  4530.2    0.07       0
  4538.4    0.05       0  4890.6     0.1       0
Bank Sta=4530.2,4538.4
Exp/Cntr=0.3,0.1

Type RM Length L Ch R = 1,28157,233,233,233
BEGIN DESCRIPTION:
Mapping XS 16658c60
END DESCRIPTION:
XS GIS Cut Line= 4
      1961016.10     13547496.65      1960641.11     13546283.11
      1960497.88     13545806.55      1960445.80     13545712.82
#Sta/Elev= 30
  3626.4  619.22  3889.8  615.34  4304.2  612.22  4517.8  609.11  4748.0  610.06
  4881.1  609.29  4896.0  608.88  4896.5  608.38  4904.2  608.88  4938.4  609.76
  4966.2  609.19  4971.4  610.05  5004.4  609.14  5037.5  609.51  5042.7  610.53
  5070.5  609.31  5075.7  610.64  5108.7  609.24  5114.0  610.65  5141.8  609.34
  5147.0  610.98  5174.8  609.61  5180.0  611.10  5213.1  610.11  5218.3  611.07
  5246.1  610.70  5251.3  611.55  5279.1  611.04  5343.6  613.36  5501.4  622.46
#Mann=5,-1,0
  3626.4     0.1       0  4304.2    0.05       0  4881.1     0.1       0
  4896.0    0.07       0  4904.2     0.1       0
Bank Sta=4896,4904.2
Exp/Cntr=0.3,0.1

Type RM Length L Ch R = 1,27924,621,621,621
BEGIN DESCRIPTION:
Horse Creek 21.0
END DESCRIPTION:
XS GIS Cut Line= 3
      1961437.99     13547285.74      1960825.00     13546125.00
      1960589.51     13545635.68
#Sta/Elev= 30
  3698.4  618.27  3864.3  615.10  3902.7  614.86  3914.1  615.64  3936.7  614.19
  4114.1  612.25  4331.7  609.59  4403.4  609.43  4425.4  610.11  4456.9  609.20
  4524.2  609.82  4536.1  608.94  4671.8  607.16  4728.3  608.15  4826.8  607.25
  4934.1  607.42  4980.9  608.28  4993.1  606.36  4993.6  605.86  5001.3  606.36
  5033.3  608.47  5087.5  606.96  5099.8  608.02  5144.2  608.20  5183.5  607.09
  5279.6  609.15  5415.4  614.58  5421.7  615.48  5534.1  620.54  5554.1  622.42
#Mann=5,-1,0
  3698.4     0.1       0  4114.1    0.05       0  4934.1     0.1       0
  4993.1    0.07       0  5001.3     0.1       0
Bank Sta=4993.1,5001.3
Exp/Cntr=0.3,0.1

Type RM Length L Ch R = 1,27303,99,99,99
BEGIN DESCRIPTION:
Horse Creek 20.0
END DESCRIPTION:
XS GIS Cut Line= 4
      1962160.42     13546941.67      1961702.10     13546066.68
      1961224.87     13545942.84      1960701.45     13545552.22
#Sta/Elev= 30
  3261.7  616.33  3373.4  614.12  3432.2  611.76  3545.4  610.59  3731.6  607.95
  3905.9  607.03  4101.0  605.28  4150.8  605.84  4227.8  604.09  4233.4  604.79
  4294.0  604.03  4294.5  603.53  4302.2  604.03  4431.3  605.27  4715.3  605.58
  4739.8  606.79  4744.9  606.79  4747.9  605.67  4762.5  607.39  4768.7  606.45
  4797.9  605.64  4812.5  607.18  4818.8  606.07  4854.6  605.51  4903.1  606.57
  5004.4  606.23  5127.3  609.29  5262.9  613.74  5348.3  618.43  5395.6  619.99
#Mann=7,-1,0
  3261.7     0.1       0  3432.2    0.05       0  3545.4     0.1       0
  3905.9    0.05       0  4294.0    0.07       0  4302.2    0.05       0
  4903.1     0.1       0
Bank Sta=4294,4302.2
Exp/Cntr=0.3,0.1

Type RM Length L Ch R = 1,27204,1020,1020,1020
BEGIN DESCRIPTION:
Horse Creek 19.0
END DESCRIPTION:
XS GIS Cut Line= 4
      1962219.44     13546875.67      1961729.87     13546007.65
      1961169.75     13545829.99      1960816.76     13545458.82
#Sta/Elev= 30
  3338.5  614.93  3432.8  613.18  3555.8  610.70  3929.8  607.15  4268.6  604.35
  4322.5  602.81  4323.0  602.31  4330.8  602.81  4333.6  604.17  4476.6  605.40
  4936.6  606.31  4950.8  604.97  4979.1  606.08  4996.8  603.25  5021.6  606.89
  5056.8  606.01  5205.6  610.47  5261.9  614.48  5269.1  616.51  5276.0  616.02
  5283.3  618.04  5290.2  617.46  5297.4  619.68  5304.3  618.85  5311.6  620.71
  5318.5  619.96  5339.9  622.27  5361.0  621.18  5382.4  623.97  5434.9  625.06
#Mann=7,-1,0
  3338.5     0.1       0  3432.8    0.05       0  3555.8     0.1       0
  3929.8    0.05       0  4322.5    0.07       0  4330.8    0.05       0
  4996.8     0.1       0
Bank Sta=4322.5,4330.8
Exp/Cntr=0.3,0.1

Type RM Length L Ch R = 1,26184,676,676,676
BEGIN DESCRIPTION:
Horse Creek 18.0
END DESCRIPTION:
XS GIS Cut Line= 3
      1962456.63     13546817.80      1962149.35     13545817.84
      1961575.02     13545325.02
#Sta/Elev= 30
  3505.8  613.96  3571.5  613.01  3591.8  613.83  3597.1  612.54  3613.3  612.12
  3868.5  607.32  3990.0  605.80  4031.8  606.55  4038.0  605.58  4126.0  604.95
  4167.8  605.61  4251.5  603.20  4324.7  602.54  4342.9  601.43  4451.5  600.36
  4621.2  602.19  4635.4  603.14  4656.3  602.20  4783.6  603.11  4827.9  602.78
  4961.4  603.05  4989.9  600.15  4992.3  599.08  4992.8  598.58  5000.1  598.58
  5000.6  599.08  5010.8  601.88  5082.1  604.74  5174.3  610.45  5308.7  624.35
#Mann=5,-1,0
  3505.8     0.1       0  3868.5    0.05       0  4827.9     0.1       0
  4992.3    0.07       0  5000.6     0.1       0
Bank Sta=4992.3,5000.6
Exp/Cntr=0.3,0.1

Type RM Length L Ch R = 1,25508,469,469,469
BEGIN DESCRIPTION:
Mapping XS b7a650f2
END DESCRIPTION:
XS GIS Cut Line= 4
      1962628.53     13546619.89      1962777.83     13545998.39
      1962159.77     13545213.67      1961670.22     13545005.35
#Sta/Elev= 30
  3576.9  610.92  3716.2  609.25  3865.2  606.00  4256.6  600.74  4277.4  601.74
  4348.0  601.46  4426.6  599.22  4619.0  600.16  4640.5  601.06  4647.9  600.09
  4654.2  600.85  4683.1  600.15  4697.6  600.90  4704.1  600.00  4732.8  599.87
  4747.3  600.57  4811.4  599.97  4960.2  600.93  4975.0  600.66  4983.1  599.49
  4989.4  600.10  4992.7  598.42  4993.2  597.92  5001.0  598.42  5053.6  601.33
  5138.5  600.44  5301.3  603.51  5415.8  606.66  5513.6  611.11  5747.0  618.32
#Mann=5,-1,0
  3576.9     0.1       0  3865.2    0.05       0  4960.2     0.1       0
  4992.7    0.07       0  5001.0     0.1       0
Bank Sta=4992.7,5001
Exp/Cntr=0.3,0.1

Type RM Length L Ch R = 1,25039,1845,1845,1845
BEGIN DESCRIPTION:
Horse Creek 15.0
END DESCRIPTION:
XS GIS Cut Line= 3
      1962993.93     13546330.08      1962853.35     13545256.20
      1961511.30     13544405.49
#Sta/Elev= 30
  3428.4  606.78  3685.2  602.15  4063.2  598.34  4129.4  597.77  4153.3  595.88
  4179.8  597.99  4232.2  598.26  4391.6  597.18  4427.8  595.44  4428.3  594.94
  4436.1  595.44  4463.7  597.06  4547.5  597.38  4629.9  597.88  4741.3  598.19
  4822.6  598.63  4852.8  597.20  4937.8  599.55  4974.2  597.06  4989.5  598.22
  4995.4  595.98  5004.7  596.16  5010.7  598.65  5018.6  599.65  5083.5  601.42
  5120.0  604.35  5214.0  609.13  5344.5  613.89  5590.2  612.07  6100.4  612.92
#Mann=7,-1,0
  3428.4    0.05       0  4063.2     0.1       0  4427.8    0.07       0
  4436.1     0.1       0  4547.5     0.1       0  4629.9    0.05       0
  4741.3     0.1       0
Bank Sta=4427.8,4436.1
Exp/Cntr=0.3,0.1

Type RM Length L Ch R = 1,23194,760,760,760
BEGIN DESCRIPTION:
Horse Creek 14.0
END DESCRIPTION:
XS GIS Cut Line= 3
      1964994.67     13545750.93      1963538.24     13544761.41
      1961815.16     13543572.18
#Sta/Elev= 30
  3336.9  618.80  3412.4  615.94  3514.1  615.98  3693.8  612.03  3966.3  601.50
  4321.2  594.48  4406.3  593.17  4730.1  594.09  4846.5  593.51  4881.9  593.22
  4968.6  593.51  4989.0  587.58  4989.5  587.08  5003.3  587.58  5004.9  590.05
  5011.1  592.19  5017.1  590.24  5026.0  592.87  5041.0  593.43  5479.3  594.57
  5721.8  594.29  6158.8  600.11  6716.6  604.70  6724.9  604.63  6906.8  604.89
  6936.7  607.39  7032.1  608.81  7067.5  611.00  7088.7  611.91  7191.3  616.25
#Mann=14,-1,0
  3336.9     0.1       0  4321.2    0.05       0  4730.1     0.1       0
  4846.5    0.05       0  4881.9     0.1       0  4989.0    0.07       0
  5003.3     0.1       0  5479.3    0.05       0  6158.8     0.1       0
  6716.6    0.12       0  6724.9    0.08       0  6906.8     0.1       0
  7067.5    0.05       0  7088.7     0.1       0
Bank Sta=4989,5003.3
Exp/Cntr=0.3,0.1

Type RM Length L Ch R = 1,22434,995,995,995
BEGIN DESCRIPTION:
Mapping XS 1c3d2587
END DESCRIPTION:
XS GIS Cut Line= 4
      1965460.11     13545756.19      1965111.16     13544902.04
      1963475.74     13544131.20      1962184.11     13543527.05
#Sta/Elev= 30
  2849.8  610.99  3032.3  605.64  3313.3  601.87  4188.2  595.34  4450.0  592.88
  4464.7  592.69  4630.5  588.81  4828.4  591.35  4962.2  590.71  4976.1  589.10
  4977.2  586.71  4977.7  586.21  4991.5  586.71  5006.4  590.15  5021.7  591.19
  5092.2  590.95  5194.3  591.65  5328.9  589.08  5625.2  592.97  5744.9  591.57
  5773.3  593.26  5819.0  592.48  5933.2  594.94  6081.3  594.17  6472.2  601.74
  6554.6  603.39  6594.8  602.08  6652.1  604.95  6925.6  609.94  7006.4  613.64
#Mann=9,-1,0
  2849.8     0.1       0  3313.3    0.05       0  4188.2     0.1       0
  4450.0    0.05       0  4464.7     0.1       0  4977.2    0.07       0
  4991.5     0.1       0  5092.2    0.05       0  6472.2     0.1       0
Bank Sta=4977.2,4991.5
Exp/Cntr=0.3,0.1

Type RM Length L Ch R = 1,21439,162,162,162
BEGIN DESCRIPTION:
Horse Creek 10.0
END DESCRIPTION:
XS GIS Cut Line= 4
      1967024.98     13545424.98      1965850.74     13544198.91
      1963309.08     13543943.70      1962224.99     13543425.00
#Sta/Elev= 30
  1885.3  612.52  2238.9  599.11  2985.7  592.88  3056.5  592.99  3371.4  591.79
  4895.3  588.09  4972.0  587.76  4977.0  587.43  4978.0  584.74  4978.5  584.24
  4993.5  584.74  5086.2  589.73  5106.3  585.62  5116.4  585.53  5126.4  587.45
  5287.2  590.63  5317.4  586.47  5337.5  588.83  5378.2  589.54  5568.6  587.14
  5578.8  588.94  5665.3  589.50  5740.6  590.82  5866.5  591.33  6333.6  594.44
  6559.3  598.41  6792.6  602.81  6888.8  606.91  7160.9  612.64  7339.2  618.81
#Mann=11,-1,0
  1885.3     0.1       0  2985.7    0.05       0  3056.5     0.1       0
  3371.4    0.05       0  4895.3     0.1       0  4978.0    0.07       0
  4993.5     0.1       0  5665.3    0.05       0  5740.6    0.08       0
  5866.5    0.05       0  6559.3     0.1       0
Bank Sta=4978,4993.5
Exp/Cntr=0.3,0.1

Type RM Length L Ch R = 1,21277,1809,1809,1809
BEGIN DESCRIPTION:
Mapping XS f75e9110
END DESCRIPTION:
XS GIS Cut Line= 4
      1967142.41     13545349.96      1965991.37     13544042.66
      1963298.66     13543797.87      1962579.93     13543386.42
#Sta/Elev= 30
  1721.3  610.88  1992.5  598.93  2084.6  596.70  2289.5  595.95  2389.1  593.73
  2898.7  592.01  3458.2  588.88  4487.7  589.79  4911.3  586.69  4935.5  586.63
  4955.6  583.88  4975.7  587.08  4985.7  585.67  4988.0  582.52  4988.5  582.02
  5003.5  582.52  5005.8  585.58  5015.9  586.79  5116.3  589.12  5216.7  589.77
  5255.8  585.41  5260.8  588.70  5317.1  589.70  5476.7  587.65  5587.2  590.55
  5813.1  590.78  6303.6  595.30  6516.8  598.69  6905.1  610.79  6995.1  611.45
#Mann=5,-1,0
  1721.3     0.1       0  2898.7    0.05       0  4911.3     0.1       0
  4988.0    0.07       0  5003.5     0.1       0
Bank Sta=4988,5003.5
Exp/Cntr=0.3,0.1

Type RM Length L Ch R = 1,19468,1832,1832,1832
BEGIN DESCRIPTION:
Horse Creek 9.0
END DESCRIPTION:
XS GIS Cut Line= 6
      1967275.03     13545325.04      1965991.87     13543891.41
      1965870.71     13543756.03      1965492.24     13543641.45
      1964772.62     13542714.54      1964625.00     13541724.97
#Sta/Elev= 30
  1530.8  609.24  1693.4  603.03  1729.4  600.14  1941.7  595.38  2239.3  592.66
  2771.6  590.56  3386.1  587.59  4018.6  587.81  4682.9  585.24  4812.2  583.43
  4967.8  583.62  4982.3  582.31  4989.0  578.59  4989.5  578.09  5004.5  578.59
  5011.3  584.90  5121.4  583.82  5175.1  582.92  5275.7  584.53  5295.9  583.79
  5326.2  579.70  5336.4  583.23  5359.6  584.60  5557.9  584.48  5680.1  586.08
  6023.9  595.40  6107.0  600.49  6135.1  603.45  6171.2  609.59  6205.9  612.71
#Mann=7,-1,0
  1530.8     0.1       0  2771.6    0.05       0  4682.9     0.1       0
  4989.0    0.07       0  5004.5     0.1       0  5121.4    0.12       0
  5359.6     0.1       0
Bank Sta=4989,5004.5
Exp/Cntr=0.3,0.1

Type RM Length L Ch R = 1,17636,744,744,744
BEGIN DESCRIPTION:
Horse Creek 8.0
END DESCRIPTION:
XS GIS Cut Line= 4
      1967425.01     13545225.03      1966808.21     13543537.28
      1965579.04     13541947.00      1964524.98     13541424.99
#Sta/Elev= 30
  1456.4  605.32  1613.7  597.83  1775.8  594.12  2454.6  587.47  2563.7  585.19
  2616.9  586.43  3188.2  583.93  3677.6  584.83  4615.5  581.90  4754.4  579.37
  4961.7  579.58  4988.9  578.10  4994.5  573.65  4995.0  573.15  5012.3  573.65
  5017.9  578.00  5032.4  579.67  5379.4  578.16  5926.2  587.67  5970.8  590.45
  6044.2  598.32  6072.2  599.30  6133.9  606.85  6139.5  605.60  6178.8  608.21
  6184.4  606.72  6251.7  605.36  6318.9  609.86  6403.1  620.07  6439.5  621.54
#Mann=5,-1,0
  1456.4     0.1       0  2454.6    0.05       0  4615.5     0.1       0
  4994.5    0.07       0  5012.3     0.1       0
Bank Sta=4994.5,5012.3
Exp/Cntr=0.3,0.1

Type RM Length L Ch R = 1,16892,1432,1432,1432
BEGIN DESCRIPTION:
Horse Creek 7.0
END DESCRIPTION:
XS GIS Cut Line= 3
      1968125.00     13544975.00      1966325.00     13541975.00
      1965124.99     13541174.99
#Sta/Elev= 30
  1519.9  601.52  1766.7  596.36  2031.1  588.84  2627.8  583.81  2649.5  582.57
  2709.2  583.37  3335.3  581.64  4027.2  582.87  4713.3  580.64  4885.7  578.55
  4967.9  577.88  4983.5  576.08  4986.1  574.02  4986.6  573.52  5004.1  574.02
  5010.7  576.62  5026.0  577.87  5117.1  577.29  5140.2  575.62  5162.7  577.45
  5206.3  577.53  5371.5  576.05  5437.6  577.14  5458.6  576.03  5596.3  578.50
  5969.4  581.21  6230.8  586.63  6330.0  588.96  6396.1  595.55  6460.7  597.67
#Mann=8,-1,0
  1519.9     0.1       0  2649.5    0.08       0  2709.2    0.05       0
  4885.7     0.1       0  4986.1    0.07       0  5004.1     0.1       0
  5117.1    0.05       0  5596.3     0.1       0
Bank Sta=4986.1,5004.1
Exp/Cntr=0.3,0.1

Type RM Length L Ch R = 1,15460,1389,1389,1389
BEGIN DESCRIPTION:
Mapping XS 7ccfb732
END DESCRIPTION:
XS GIS Cut Line= 4
      1969161.94     13544193.53      1967851.18     13541493.88
      1966227.91     13540677.90      1965508.68     13539854.69
#Sta/Elev= 30
  1016.0  590.03  1837.2  580.02  1948.5  579.47  2059.8  578.76  2474.8  576.32
  2838.8  576.27  2885.5  576.60  2932.9  576.67  3174.0  577.05  4144.7  575.53
  4803.4  573.25  4825.7  571.15  4937.3  574.68  4982.0  574.24  4987.6  573.06
  4988.6  569.98  4989.1  569.48  5006.7  569.98  5009.9  573.70  5020.1  574.58
  5339.2  572.53  5753.3  578.59  5866.0  581.06  5944.0  579.28  6277.0  591.22
  6390.9  600.38  6475.4  611.86  6525.7  611.62  6595.9  616.66  6927.0  620.61
#Mann=14,-1,0
  1016.0     0.1       0  1837.2    0.08       0  1948.5    0.05       0
  2059.8     0.1       0  2474.8    0.05       0  2838.8     0.1       0
  2885.5    0.05       0  2932.9     0.1       0  3174.0    0.05       0
  4144.7     0.1       0  4988.6    0.07       0  5006.7     0.1       0
  5753.3    0.05       0  5944.0     0.1       0
Bank Sta=4988.6,5006.7
Exp/Cntr=0.3,0.1

Type RM Length L Ch R = 1,14071,950,950,950
BEGIN DESCRIPTION:
Mapping XS 0782ced8
END DESCRIPTION:
XS GIS Cut Line= 4
      1969361.59     13543967.82      1968458.82     13541632.77
      1967078.61     13539566.79      1966210.52     13538993.86
#Sta/Elev= 30
   723.5  586.67  1423.7  579.39  1590.0  577.83  2079.7  574.68  2223.5  574.62
  2452.8  574.68  2625.8  574.58  3214.4  574.34  3819.8  574.06  3867.6  573.73
  4338.8  567.48  4483.0  570.36  4581.8  567.19  4582.3  566.69  4600.4  567.19
  4655.4  570.45  4880.3  570.02  4980.1  571.66  5002.6  568.44  5029.6  571.12
  5239.9  571.43  5485.2  576.36  5636.3  582.99  5810.2  595.64  5852.4  601.33
  5939.7  605.86  6156.4  601.59  6445.4  603.58  6566.6  608.01  6751.7  605.93
#Mann=13,-1,0
   723.5     0.1       0  1423.7    0.05       0  1590.0     0.1       0
  2079.7    0.05       0  2223.5     0.1       0  2452.8    0.05       0
  2625.8     0.1       0  3214.4    0.05       0  3819.8     0.1       0
  3867.6    0.05       0  4581.8    0.07       0  4600.4    0.05       0
  4880.3     0.1       0
Bank Sta=4581.8,4600.4
Exp/Cntr=0.3,0.1

Type RM Length L Ch R = 1,13121,279,279,279
BEGIN DESCRIPTION:
Mapping XS 6c6886f4
END DESCRIPTION:
XS GIS Cut Line= 2
      1969613.33     13543898.39      1967486.60     13538160.55
#Sta/Elev= 30
   586.1  586.00  1356.3  578.08  1456.3  577.03  1461.6  576.96  1973.8  573.30
  3908.2  572.03  3970.5  569.38  4110.2  570.24  4165.7  567.78  4237.1  569.39
  4290.4  565.84  4453.5  570.14  4962.3  569.11  4973.8  568.89  4984.1  565.36
  4984.6  564.86  5002.9  565.36  5036.9  568.93  5079.3  569.64  5115.0  567.36
  5122.3  569.73  5164.9  567.72  5170.4  569.67  5175.8  567.74  5195.5  570.18
  5250.2  571.12  5483.3  572.61  5538.2  575.06  6455.4  587.36  6705.4  598.00
#Mann=6,-1,0
   586.1     0.1       0  1356.3    0.08       0  1456.3    0.05       0
  1461.6     0.1       0  4984.1    0.07       0  5002.9     0.1       0
Bank Sta=4984.1,5002.9
Exp/Cntr=0.3,0.1

Type RM Length L Ch R = 1,12842,1625,1625,1625
BEGIN DESCRIPTION:
Mapping XS 2e80a77e
END DESCRIPTION:
XS GIS Cut Line= 2
      1969804.30     13543724.79      1967816.46     13538230.01
#Sta/Elev= 30
   718.0  582.43  1043.2  580.49  1089.8  579.99  1240.4  578.57  1398.5  577.03
  1575.1  575.57  1610.6  575.79  2121.5  571.06  2558.0  572.83  2873.9  570.61
  3878.7  570.95  4261.2  568.53  4369.1  563.15  4369.6  562.65  4387.9  563.15
  4418.5  567.06  4535.5  568.82  4854.5  569.15  4934.2  566.46  4964.9  568.06
  5003.4  564.93  5020.8  568.22  5067.2  569.92  5120.4  568.16  5481.9  572.44
  5769.1  580.20  6137.7  594.70  6310.9  596.10  6408.2  593.86  6561.3  595.91
#Mann=9,-1,0
   718.0     0.1       0  1043.2    0.08       0  1089.8     0.1       0
  1240.4    0.08       0  1398.5     0.1       0  1575.1    0.08       0
  1610.6     0.1       0  4369.1    0.07       0  4387.9     0.1       0
Bank Sta=4369.1,4387.9
Exp/Cntr=0.3,0.1

Type RM Length L Ch R = 1,11217,1021,1021,1021
BEGIN DESCRIPTION:
Horse Creek 3.0
END DESCRIPTION:
XS GIS Cut Line= 3
      1969301.18     13540900.18      1969061.61     13538962.72
      1968484.30     13537948.54
#Sta/Elev= 30
  3210.1  570.15  3900.5  566.11  3961.0  561.04  4021.4  565.73  4202.8  566.40
  4243.1  563.58  4253.8  559.45  4254.3  558.95  4272.7  559.45  4278.7  563.40
  4293.5  565.83  4323.7  566.16  4484.9  565.38  4521.8  561.81  4526.9  563.46
  4545.4  562.50  4565.5  565.73  4807.4  565.31  4837.6  567.11  4932.1  563.20
  4958.5  565.30  4988.7  563.95  4998.8  561.17  5019.0  564.11  5165.5  564.52
  5620.0  573.24  5746.3  578.76  5832.7  585.40  6103.2  580.59  6329.3  584.28
#Mann=3,-1,0
  3210.1     0.1       0  4253.8    0.07       0  4272.7     0.1       0
Bank Sta=4253.8,4272.7
Exp/Cntr=0.3,0.1

Type RM Length L Ch R = 1,10196,1905,1905,1905
BEGIN DESCRIPTION:
Horse Creek 2.0
END DESCRIPTION:
XS GIS Cut Line= 3
      1969848.06     13540905.39      1969889.73     13538764.81
      1968947.01     13537410.62
#Sta/Elev= 30
  3168.8  567.30  3549.3  565.73  3699.3  562.86  3879.3  562.10  3909.3  559.10
  3939.3  562.50  4102.3  563.23  4252.1  563.19  4369.4  562.81  4399.4  561.04
  4449.4  562.41  4459.4  560.09  4460.0  558.12  4460.5  557.62  4478.9  558.12
  4479.4  560.32  4519.4  563.43  4839.5  562.99  4989.5  561.05  4999.5  559.31
  5009.5  559.45  5019.5  562.08  5289.6  560.55  5622.3  564.63  5637.2  563.57
  5953.1  569.98  6161.7  570.28  6406.0  573.32  6491.5  576.31  6959.8  584.58
#Mann=5,-1,0
  3168.8     0.1       0  4102.3    0.16       0  4252.1     0.1       0
  4460.0    0.07       0  4478.9     0.1       0
Bank Sta=4460,4478.9
Exp/Cntr=0.3,0.1

Type RM Length L Ch R = 1,8291,1144,1144,1144
BEGIN DESCRIPTION:
Mapping XS 7c7e0425
END DESCRIPTION:
XS GIS Cut Line= 4
      1970535.55     13540491.83      1970910.56     13539767.85
      1970863.69     13538278.26      1970223.05     13537252.20
#Sta/Elev= 30
  3357.2  562.98  3600.9  561.21  3689.4  559.49  3702.7  557.20  3761.5  561.15
  3778.0  566.33  3783.6  563.15  3800.1  566.69  3805.7  563.30  3822.2  565.34
  3827.9  560.97  3848.8  559.72  3923.1  559.75  4006.8  561.94  4015.8  559.95
  4096.9  559.41  4148.6  554.96  4164.5  559.18  4190.4  560.23  4798.7  557.37
  4855.7  555.55  4975.8  558.55  4985.8  558.37  4986.2  554.47  4986.7  553.97
  5005.3  554.47  5020.9  558.43  5173.4  557.94  5926.1  562.53  6872.5  575.09
#Mann=8,-1,0
  3357.2     0.1       0  3848.8    0.16       0  3923.1     0.1       0
  4798.7    0.12       0  4986.2    0.07       0  5005.3    0.12       0
  5020.9    0.16       0  5173.4     0.1       0
Bank Sta=4986.2,5005.3
Exp/Cntr=0.3,0.1

Type RM Length L Ch R = 1,7147,1081,1081,1081
BEGIN DESCRIPTION:
Mapping XS d068736f
END DESCRIPTION:
XS GIS Cut Line= 4
      1971493.90     13541002.21      1971447.02     13539679.30
      1971572.02     13538523.05      1970894.95     13537330.36
#Sta/Elev= 30
  3246.6  562.26  3734.1  556.19  3864.4  556.28  3914.2  556.04  3944.3  552.26
  3964.0  553.38  4024.3  555.96  4044.3  553.37  4074.3  557.18  4114.4  557.76
  4464.6  555.66  4799.9  557.35  4886.5  557.45  4977.0  555.01  4987.1  553.85
  4987.5  550.93  4988.0  550.43  5006.7  550.93  5017.2  554.17  5097.7  553.77
  5159.7  558.33  5319.0  564.69  5671.0  571.25  5765.6  571.60  6060.2  565.78
  6264.9  563.66  6280.8  564.99  6339.9  564.14  6733.6  568.29  7104.8  570.01
#Mann=6,-1,0
  3246.6     0.1       0  3864.4    0.12       0  3964.0     0.1       0
  4799.9    0.12       0  4987.5    0.07       0  5006.7     0.1       0
Bank Sta=4987.5,5006.7
Exp/Cntr=0.3,0.1
