--- UNT 001 in BCW.prj (project) ---

Proj Title=UNT 001 in BCW Base Level Engineering
Current Plan=p01
Default Exp/Contr=0.3,0.1
English Units
Geom File=g01
Flow File=f01
Plan File=p01
Y Axis Title=Elevation
X Axis Title(PF)=Main Channel Distance
X Axis Title(XS)=Station
BEGIN DESCRIPTION:
UNT 001 in BCW
END DESCRIPTION:
DSS File=dss
DSS Export Rating Curves= 0
DSS Export Rating Curve Sorted= 0
DSS Export Volume Flow Curves= 0
DXF OffsetX= 0
DXF OffsetY= 0
DXF ScaleX= 1
DXF ScaleY= 10

--- UNT 001 in BCW.p01 (plan) ---

Plan Title=Multiple Run
Program Version=5.05
Short Identifier=Multiple Run
Geom File=g01
Flow File=f01
Subcritical Flow
K Sum by GR= 0
Std Step Tol= 0.01
Critical Tol= 0.01
Num of Std Step Trials= 20
Max Error Tol= 0.3
Flow Tol Ratio= 0.001
Split Flow NTrial= 30
Split Flow Tol= 0.02
Split Flow Ratio= 0.02
Log Output Level= 0
Friction Slope Method= 1
Unsteady Friction Slope Method= 2
Unsteady Bridges Friction Slope Method= 1
Parabolic Critical Depth
Global Vel Dist= 1 , 1 , 1
Global Log Level= 0
CheckData=True
Encroach Param=-1 ,0,0, 0
BEGIN DESCRIPTION:
Multiple Run
END DESCRIPTION:
Computation Interval=1MIN
Output Interval=1HOUR
Instantaneous Interval=1HOUR
Mapping Interval=1HOUR
Computation Time Step Use Courant=        0
Computation Time Step Use Time Series=    0
Computation Time Step Count To Double=0
Computation Time Step Max Doubling=0
Computation Time Step Max Halving=0
Computation Time Step Residence Courant=0
Run HTab= 0
Run UNet= 0
Run Sediment= 0
Run PostProcess= 0
Run WQNet= 0
Run RASMapper= 0
UNET Theta= 1
UNET Theta Warmup= 1
UNET ZTol= 0.02
UNET ZSATol= 0.02
UNET MxIter= 20
UNET Max Iter WO Improvement= 0
UNET MaxInSteps= 0
UNET DtIC= 0
UNET DtMin= 0
UNET MaxCRTS= 20
UNET WFStab= 2
UNET SFStab= 1
UNET WFX= 1
UNET SFX= 1
UNET 1D Methodology=Finite Difference
UNET DSS MLevel= 4
UNET Pardiso=0
UNET DZMax Abort= 100
UNET Use Existing IB Tables=-1
UNET Froude Reduction=False
UNET Froude Limit= 0.8
UNET Froude Power= 4
UNET D1 Cores= 0
UNET D2 Coriolis=0
UNET D2 Cores= 0
UNET D2 Theta= 1
UNET D2 Theta Warmup= 1
UNET D2 Z Tol= 0.01
UNET D2 Volume Tol= 0.01
UNET D2 Max Iterations= 20
UNET D2 Equation= 0
UNET D2 RampUpFraction=0.1
UNET D2 TimeSlices= 1
UNET D2 BCVolumeCheck=0
UNET D1D2 MaxIter= 0
UNET D1D2 ZTol=0.01
UNET D1D2 QTol=0.1
UNET D1D2 MinQTol=1
DSS File=dss
Write IC File= 0
Write IC File at Fixed DateTime=0
Write IC File at Sim End=0
Echo Input=False
Echo Parameters=False
Echo Output=False
Write Detailed= 0
HDF Write Warmup=0
HDF Write Time Slices=0
HDF Flush=0
HDF Face Node Velocities=0
HDF Compression= 1
HDF Chunk Size= 1
HDF Spatial Parts= 1
HDF Use Max Rows=0
HDF Fixed Rows= 1
Calibration Method= 0
Calibration Iterations= 20
Calibration Max Change=0.05
Calibration Tolerance=0.2
Calibration Maximum=1.5
Calibration Minimum=0.5
Calibration Optimization Method= 1
WQ AD Non Conservative
WQ ULTIMATE=-1
WQ Max Comp Step=1HOUR
WQ Output Interval=15MIN
WQ Output Selected Increments= 0
WQ Output face flow=0
WQ Output face velocity=0
WQ Output face area=0
WQ Output face dispersion=0
WQ Output cell volume=0
WQ Output cell surface area=0
WQ Output cell continuity=0
WQ Output cumulative cell continuity=0
WQ Output face conc=0
WQ Output face dconc_dx=0
WQ Output face courant=0
WQ Output face peclet=0
WQ Output face adv mass=0
WQ Output face disp mass=0
WQ Output cell mass=0
WQ Output cell source sink temp=0
WQ Output nsm pathways=0
WQ Output nsm derived pathways=0
WQ Output MaxMinRange=-1
WQ Daily Max Min Mean=-1
WQ Daily Range=0
WQ Daily Time=0
WQ Create Restart=0
WQ Fixed Restart=0
WQ System Summary=0
WQ Write To DSS=0
WQ Use Fixed Temperature=0
Sorting and Armoring Iterations= 10
XS Update Threshold= 0.02
Bed Roughness Predictor= 0
Hydraulics Update Threshold= 0.02
Energy Slope Method= 1
Volume Change Method= 1
Sediment Retention Method= 0
XS Weighting Method= 0
Number of US Weighted Cross Sections= 1
Number of DS Weighted Cross Sections= 1
Upstream XS Weight=0
Main XS Weight=1
Downstream XS Weight=0
Number of DS XS's Weighted with US Boundary= 1
Upstream Boundary Weight= 1
Weight of XSs Associated with US Boundary= 0
Number of US XS's Weighted with DS Boundary= 1
Downstream Boundary Weight= 0.5
Weight of XSs Associated with DS Boundary= 0.5
Percentile Method= 0
Sediment Output Level= 3
Mass or Volume Output= 0
Output Increment Type= 1
Profile and TS Output Increment= 1
XS Output Flag= 0
XS Output Increment= 10
Write Gradation File= 0
Read Gradation Hotstart= 0
Write HDF5 File= 1
Write Binary Output= 1
Write DSS Sediment File= 0
SV Curve= 0
Specific Gage Flag= 0

--- UNT 001 in BCW.f01 (steady flow) ---

Flow Title=Multiple
Program Version=5.05
Number of Profiles= 7
Profile Names=10-year,25-year,50-year,1pct_min,100-year,1pct_plu,500-year
River Rch & RM=UNT 001 in BCW,Reach-1         ,22876
     150     206     252     155     309     617     473
River Rch & RM=UNT 001 in BCW,Reach-1         ,22564
     159     219     268     165     329     655     502
River Rch & RM=UNT 001 in BCW,Reach-1         ,20248
     224     313     388     241     480     958     747
River Rch & RM=UNT 001 in BCW,Reach-1         ,17076
     343     489     613     384     767    1530    1221
River Rch & RM=UNT 001 in BCW,Reach-1         ,16198
     477     685     864     543    1083    2161    1733
River Rch & RM=UNT 001 in BCW,Reach-1         ,5493
     619     898    1139     719    1434    2862    2317
River Rch & RM=UNT 001 in BCW,Reach-1         ,2362
     641     929    1179     744    1485    2962    2397
Boundary for River Rch & Prof#=UNT 001 in BCW,Reach-1         , 1
Up Type= 0
Dn Type= 3
Dn Slope=0.00467
Boundary for River Rch & Prof#=UNT 001 in BCW,Reach-1         , 2
Up Type= 0
Dn Type= 3
Dn Slope=0.00467
Boundary for River Rch & Prof#=UNT 001 in BCW,Reach-1         , 3
Up Type= 0
Dn Type= 3
Dn Slope=0.00467
Boundary for River Rch & Prof#=UNT 001 in BCW,Reach-1         , 4
Up Type= 0
Dn Type= 3
Dn Slope=0.00467
Boundary for River Rch & Prof#=UNT 001 in BCW,Reach-1         , 5
Up Type= 0
Dn Type= 3
Dn Slope=0.00467
Boundary for River Rch & Prof#=UNT 001 in BCW,Reach-1         , 6
Up Type= 0
Dn Type= 3
Dn Slope=0.00467
Boundary for River Rch & Prof#=UNT 001 in BCW,Reach-1         , 7
Up Type= 0
Dn Type= 3
Dn Slope=0.00467
DSS Import GetInterval= 0
DSS Import GetPeak= 0
DSS Import FillOption= 0

--- UNT 001 in BCW.g01 (geometry) ---

Geom Title=Existing Conditions

River Reach=UNT 001 in BCW,Reach-1
Reach XY= 30
      1961152.54     13482506.64      1963290.80     13483594.54
      1963790.80     13484084.54      1964230.80     13484164.54
      1964400.80     13484324.54      1964740.80     13484164.54
      1965258.06     13484306.25      1968470.80     13486474.54
      1969190.80     13486784.54      1969780.80     13486804.54
      1970461.01     13487364.54      1970621.60     13487865.40
      1971182.36     13488076.34      1971466.22     13488042.49
      1972211.18     13487485.98      1972801.13     13487965.35
      1973273.01     13488962.75      1973882.38     13489246.08
      1974801.91     13489285.14      1975572.75     13489597.12
      1975830.80     13489834.54      1975948.70     13490074.81
      1975828.57     13490227.59      1976213.29     13490720.64
      1976192.45     13491731.06      1976280.80     13492004.54
      1976650.80     13492264.54      1977429.40     13492391.27
      1977635.65     13492608.63      1977630.80     13493014.54

Type RM Length L Ch R = 1,22876,312,312,312
BEGIN DESCRIPTION:
UNT 001 in BCW 43.0
END DESCRIPTION:
XS GIS Cut Line= 3
      1960978.13     13482968.04      1961328.13     13482568.06
      1961627.67     13481919.04
#Sta/Elev= 30
  4527.9  595.64  4775.7  588.92  4945.6  586.75  4967.5  587.61  4993.9  584.83
  4994.2  584.33  4997.9  584.83  5010.2  586.57  5061.6  586.00  5073.8  586.76
  5095.8  585.84  5128.8  586.54  5157.8  589.53  5209.2  590.28  5294.0  589.81
  5329.5  590.62  5346.9  592.06  5352.4  591.10  5375.4  591.35  5415.2  592.75
  5426.8  594.59  5437.2  595.08  5449.7  594.42  5638.8  598.90  5707.6  601.86
  5730.6  601.33  5745.6  602.37  5753.5  604.30  5767.6  603.05  5774.2  603.34
#Mann=3,-1,0
  4527.9     0.1       0  4993.9    0.07       0  4997.9     0.1       0
Bank Sta=4993.9,4997.9
Exp/Cntr=0.3,0.1

Type RM Length L Ch R = 1,22564,600,600,600
BEGIN DESCRIPTION:
Mapping XS fff17b8e
END DESCRIPTION:
XS GIS Cut Line= 2
      1961222.80     13483205.82      1961972.80     13482112.06
#Sta/Elev= 30
  4410.7  604.30  4794.2  586.42  4823.9  586.72  4830.1  588.30  4851.0  588.23
  4880.8  586.60  4886.9  584.33  4906.8  583.42  4907.1  582.92  4910.8  583.42
  5090.0  585.78  5096.1  585.02  5125.9  585.39  5248.3  590.48  5333.2  592.15
  5391.9  596.18  5427.7  600.66  5442.3  598.47  5454.8  598.59  5469.7  601.21
  5499.5  604.04  5556.3  607.78  5571.2  611.05  5586.1  612.38  5592.2  611.58
  5607.1  615.13  5613.2  614.09  5643.0  618.70  5678.8  620.65  5736.9  620.97
#Mann=3,-1,0
  4410.7     0.1       0  4906.8    0.07       0  4910.8     0.1       0
Bank Sta=4906.8,4910.8
Exp/Cntr=0.3,0.1

Type RM Length L Ch R = 1,21964,434,434,434
BEGIN DESCRIPTION:
UNT 001 in BCW 42.0
END DESCRIPTION:
XS GIS Cut Line= 4
      1961625.01     13483324.99      1962008.11     13483030.94
      1962117.48     13482713.23      1962143.52     13482175.00
#Sta/Elev= 30
  4415.5  604.67  4522.4  592.60  4551.5  590.81  4557.8  591.44  4566.0  589.99
  4593.1  587.45  4665.7  586.16  4680.2  585.75  4692.8  584.39  4750.9  583.12
  4850.6  581.43  4879.6  581.94  4987.3  579.64  4987.5  579.14  4991.4  579.64
  5010.5  580.60  5151.6  582.45  5302.8  586.00  5402.9  589.18  5442.9  591.81
  5483.0  591.01  5503.0  593.59  5523.0  593.84  5563.1  596.50  5683.2  601.26
  5699.3  602.53  5704.3  601.87  5723.2  603.00  5743.3  602.98  5773.3  605.26
#Mann=3,-1,0
  4415.5     0.1       0  4987.3    0.07       0  4991.4     0.1       0
Bank Sta=4987.3,4991.4
Exp/Cntr=0.3,0.1

Type RM Length L Ch R = 1,21530,451,451,451
BEGIN DESCRIPTION:
UNT 001 in BCW 41.0
END DESCRIPTION:
XS GIS Cut Line= 3
      1962024.97     13483575.03      1962375.00     13483175.00
      1962775.47     13482291.36
#Sta/Elev= 30
  4433.5  595.02  4532.7  591.15  4547.0  588.65  4561.2  589.70  4575.4  589.80
  4589.7  588.30  4624.8  587.46  4667.5  585.23  4724.4  583.97  4752.4  582.52
  4837.4  580.73  4858.7  581.03  4951.3  579.93  5000.3  577.96  5000.6  577.46
  5004.3  577.46  5004.5  577.96  5019.9  579.08  5054.1  579.83  5221.2  580.20
  5440.0  583.25  5470.1  585.62  5486.2  585.99  5509.3  585.37  5612.8  590.85
  5635.8  591.10  5658.8  592.79  5820.5  599.52  5832.4  600.94  5935.2  605.70
#Mann=3,-1,0
  4433.5     0.1       0  5000.3    0.07       0  5004.5     0.1       0
Bank Sta=5000.3,5004.5
Exp/Cntr=0.3,0.1

Type RM Length L Ch R = 1,21079,476,476,476
BEGIN DESCRIPTION:
UNT 001 in BCW 40.0
END DESCRIPTION:
XS GIS Cut Line= 3
      1962375.02     13483724.98      1962775.00     13483325.00
      1962992.49     13482501.39
#Sta/Elev= 30
  4458.2  596.53  4613.7  588.72  4684.4  585.62  4726.9  584.59  4755.2  582.76
  4825.9  580.51  4967.3  577.95  4993.4  576.72  4993.7  576.22  4997.4  576.22
  4997.7  576.72  5041.4  578.54  5292.8  579.30  5447.9  583.58  5474.0  584.58
  5479.2  585.47  5489.3  585.97  5499.6  585.61  5514.3  586.36  5530.7  586.02
  5549.4  584.50  5582.4  583.79  5603.1  588.61  5613.4  590.13  5665.0  592.14
  5670.2  591.63  5716.8  593.59  5737.5  593.65  5750.7  595.05  5875.7  600.21
#Mann=3,-1,0
  4458.2     0.1       0  4993.4    0.07       0  4997.7     0.1       0
Bank Sta=4993.4,4997.7
Exp/Cntr=0.3,0.1

Type RM Length L Ch R = 1,20603,355,355,355
BEGIN DESCRIPTION:
UNT 001 in BCW 39.0
END DESCRIPTION:
XS GIS Cut Line= 3
      1962626.15     13483993.62      1963125.00     13483575.00
      1963740.84     13483021.87
#Sta/Elev= 30
  4323.1  601.63  4420.8  597.48  4441.6  597.91  4463.7  597.10  4505.4  596.92
  4562.6  595.19  4576.9  594.17  4634.1  592.84  4704.4  586.39  4726.3  585.66
  4775.9  582.05  4868.3  578.09  4917.7  576.77  4960.6  576.58  4985.9  575.38
  4986.2  574.88  4990.3  575.38  5045.0  576.56  5172.8  576.29  5257.2  577.08
  5349.9  576.12  5477.0  580.06  5512.1  581.83  5519.6  582.78  5526.3  582.23
  5576.4  583.59  5583.2  585.60  5597.4  586.79  5625.8  585.20  5802.1  590.69
#Mann=3,-1,0
  4323.1     0.1       0  4985.9    0.07       0  4990.3     0.1       0
Bank Sta=4985.9,4990.3
Exp/Cntr=0.3,0.1

Type RM Length L Ch R = 1,20248,491,491,491
BEGIN DESCRIPTION:
UNT 001 in BCW 38.0
END DESCRIPTION:
XS GIS Cut Line= 3
      1962875.01     13484274.99      1963475.00     13483675.00
      1963870.60     13483160.78
#Sta/Elev= 30
  4210.7  604.56  4224.8  604.70  4267.3  602.34  4338.0  594.28  4366.2  592.41
  4408.7  590.67  4422.8  589.44  4578.4  582.97  4606.7  581.21  4691.5  578.35
  4852.5  575.42  4992.3  574.83  5030.9  575.25  5084.6  574.65  5085.0  574.15
  5089.6  574.15  5090.0  574.65  5116.3  575.46  5166.1  575.66  5216.0  577.27
  5273.7  580.29  5301.1  582.26  5315.6  583.88  5359.2  586.65  5444.3  587.74
  5515.0  587.60  5523.2  588.48  5551.3  587.94  5658.2  590.77  5708.0  592.64
#Mann=5,-1,0
  4210.7     0.1       0  4852.5    0.05       0  4992.3     0.1       0
  5084.6    0.07       0  5090.0     0.1       0
Bank Sta=5084.6,5090
Exp/Cntr=0.3,0.1

Type RM Length L Ch R = 1,19757,393,393,393
BEGIN DESCRIPTION:
UNT 001 in BCW 37.0
END DESCRIPTION:
XS GIS Cut Line= 3
      1963227.70     13484675.94      1963775.00     13484025.00
      1964076.67     13483191.56
#Sta/Elev= 30
  4180.6  591.29  4221.4  590.35  4243.5  587.84  4257.8  586.78  4263.2  586.99
  4272.5  586.59  4292.9  585.98  4385.4  585.74  4434.7  586.16  4442.5  585.44
  4498.4  585.21  4534.6  583.33  4562.2  583.94  4584.2  582.28  4789.8  575.29
  4964.0  573.05  4964.4  572.55  4969.0  572.55  4969.4  573.05  5318.2  573.96
  5459.4  576.31  5607.3  581.30  5647.9  583.29  5663.3  583.35  5701.0  586.14
  5796.8  590.13  5805.9  591.73  5811.2  591.27  5818.0  592.56  5917.4  594.24
#Mann=6,-1,0
  4180.6    0.05       0  4263.2     0.1       0  4272.5    0.05       0
  4385.4     0.1       0  4964.0    0.07       0  4969.4     0.1       0
Bank Sta=4964,4969.4
Exp/Cntr=0.3,0.1

Type RM Length L Ch R = 1,19364,504,504,504
BEGIN DESCRIPTION:
UNT 001 in BCW 36.0
END DESCRIPTION:
XS GIS Cut Line= 3
      1963881.39     13484688.88      1964225.99     13483862.32
      1964441.98     13483219.56
#Sta/Elev= 30
  4416.0  593.18  4420.8  593.18  4431.0  591.52  4461.2  590.03  4466.7  590.36
  4485.1  588.79  4506.9  587.83  4519.7  586.25  4561.1  584.10  4604.4  582.89
  4680.2  578.29  4779.8  574.06  4864.4  572.16  4991.6  571.78  4992.1  571.28
  4996.8  571.28  4997.2  571.78  5211.1  573.05  5286.9  572.59  5513.4  573.60
  5608.0  576.37  5671.1  579.09  5688.5  578.76  5720.1  579.47  5728.8  580.45
  5791.9  582.74  5815.1  582.57  5867.8  584.22  5910.0  584.12  5989.6  587.04
#Mann=4,-1,0
  4416.0    0.05       0  4779.8     0.1       0  4991.6    0.07       0
  4997.2     0.1       0
Bank Sta=4991.6,4997.2
Exp/Cntr=0.3,0.1

Type RM Length L Ch R = 1,18860,400,400,400
BEGIN DESCRIPTION:
UNT 001 in BCW 35.0
END DESCRIPTION:
XS GIS Cut Line= 3
      1964075.00     13484775.00      1964475.00     13484375.00
      1965126.18     13483384.21
#Sta/Elev= 30
  4350.0  590.43  4392.4  589.50  4463.1  585.04  4576.3  580.45  4632.8  577.38
  4717.7  574.41  4802.5  572.34  4948.8  570.37  4949.2  569.87  4953.9  569.87
  4954.4  570.37  5026.8  570.82  5262.7  570.54  5334.5  571.43  5363.1  571.18
  5486.6  572.93  5492.6  572.46  5522.8  572.68  5549.9  573.99  5559.0  573.89
  5564.9  572.79  5573.8  574.24  5586.0  574.55  5616.2  576.82  5673.4  577.75
  5730.6  579.47  5766.8  579.50  5789.2  580.78  5875.3  583.03  6101.3  590.69
#Mann=4,-1,0
  4350.0    0.05       0  4948.8   0.035       0  4954.4    0.05       0
  5026.8     0.1       0
Bank Sta=4948.8,4954.4
Exp/Cntr=0.3,0.1

Type RM Length L Ch R = 1,18460,478,478,478
BEGIN DESCRIPTION:
UNT 001 in BCW 34.0
END DESCRIPTION:
XS GIS Cut Line= 3
      1964429.12     13485052.42      1964825.00     13484225.00
      1965530.35     13483503.28
#Sta/Elev= 30
  4091.6  588.34  4091.9  588.34  4343.3  578.53  4622.2  572.86  4765.0  570.46
  4829.3  569.62  4984.2  567.81  4991.8  567.48  4992.3  566.98  4997.6  567.48
  5215.6  569.66  5223.4  569.55  5349.4  571.00  5514.1  575.64  5617.0  578.88
  5631.1  577.92  5652.3  579.69  5659.4  578.70  5666.4  580.35  5673.6  579.53
  5737.1  583.33  5744.3  582.51  5750.6  584.01  5758.4  583.06  5765.4  584.55
  5772.6  583.33  5804.8  584.55  5884.4  588.07  5950.2  590.62  6018.0  593.09
#Mann=16,-1,0
  4091.6     0.1       0  4091.9    0.05       0  4622.2     0.1       0
  4765.0    0.05       0  4829.3     0.1       0  4984.2    0.05       0
  4991.8    0.03       0  4997.6    0.05       0  5215.6     0.1       0
  5223.4    0.05       0  5349.4     0.1       0  5514.1    0.05       0
  5750.6     0.1       0  5804.8    0.05       0  5884.4     0.1       0
  5950.2    0.05       0
Bank Sta=4991.8,4997.6
Exp/Cntr=0.3,0.1

Type RM Length L Ch R = 1,17982,381,381,381
BEGIN DESCRIPTION:
UNT 001 in BCW 33.0
END DESCRIPTION:
XS GIS Cut Line= 3
      1964856.17     13484982.15      1965275.00     13484325.00
      1965675.03     13483924.97
#Sta/Elev= 30
  4212.6  590.03  4253.8  589.38  4259.8  589.93  4290.2  588.45  4296.2  589.03
  4311.4  587.06  4332.5  587.76  4347.8  586.14  4353.7  586.72  4363.0  585.76
  4368.9  586.64  4384.2  584.09  4390.1  585.15  4405.3  583.68  4478.1  583.94
  4484.0  584.84  4499.3  584.57  4507.9  583.50  4556.8  579.89  4760.0  570.25
  4775.2  568.85  4790.3  569.46  4861.4  567.50  4941.9  567.19  5003.1  565.87
  5003.6  565.37  5009.0  565.87  5147.4  569.41  5345.4  577.18  5557.6  594.02
#Mann=4,-1,0
  4212.6     0.1       0  4507.9    0.05       0  5003.1   0.035       0
  5009.0    0.05       0
Bank Sta=5003.1,5009
Exp/Cntr=0.3,0.1

Type RM Length L Ch R = 1,17601,525,525,525
BEGIN DESCRIPTION:
UNT 001 in BCW 32.0
END DESCRIPTION:
XS GIS Cut Line= 3
      1965168.67     13484901.41      1965820.31     13484330.21
      1966070.12     13484230.28
#Sta/Elev= 30
  4441.5  588.87  4514.6  586.84  4549.7  583.65  4556.4  581.48  4613.3  578.98
  4620.9  579.76  4635.1  578.72  4641.8  576.58  4741.4  571.89  4805.0  567.08
  4851.0  567.21  5028.8  565.39  5029.3  564.89  5034.8  565.39  5121.2  568.60
  5222.6  575.38  5251.1  580.10  5258.6  584.34  5265.3  583.67  5272.9  585.58
  5279.5  584.37  5287.1  586.97  5293.8  584.77  5301.0  588.38  5307.8  589.76
  5391.6  592.91  5415.9  595.90  5499.3  601.93  5547.8  608.53  5577.1  610.84
#Mann=5,-1,0
  4441.5     0.1       0  4851.0    0.05       0  5028.8    0.03       0
  5034.8    0.05       0  5121.2     0.1       0
Bank Sta=5028.8,5034.8
Exp/Cntr=0.3,0.1

Type RM Length L Ch R = 1,17076,379,379,379
BEGIN DESCRIPTION:
UNT 001 in BCW 31.0
END DESCRIPTION:
XS GIS Cut Line= 3
      1965925.00     13485425.00      1966025.00     13484775.00
      1966170.65     13484444.52
#Sta/Elev= 30
  4337.6  589.71  4388.2  587.74  4503.3  579.11  4540.0  575.19  4629.8  570.02
  4734.0  566.12  4926.2  562.55  4961.0  562.21  4961.5  561.71  4971.3  562.21
  5004.2  562.50  5017.1  564.25  5033.0  567.09  5039.0  571.68  5056.3  577.24
  5061.8  577.21  5079.6  582.88  5085.1  582.32  5102.9  585.09  5108.4  583.90
  5126.3  585.79  5131.7  584.65  5155.1  587.47  5160.5  586.39  5178.4  587.97
  5183.9  586.76  5201.7  587.73  5207.2  586.06  5282.6  591.45  5356.4  598.49
#Mann=5,-1,0
  4337.6     0.1       0  4734.0    0.05       0  4926.2     0.1       0
  4961.0    0.07       0  4971.3     0.1       0
Bank Sta=4961,4971.3
Exp/Cntr=0.3,0.1

Type RM Length L Ch R = 1,16697,499,499,499
BEGIN DESCRIPTION:
UNT 001 in BCW 30.0
END DESCRIPTION:
XS GIS Cut Line= 3
      1966003.77     13485546.34      1966275.00     13485075.00
      1966424.77     13484700.01
#Sta/Elev= 30
  4420.6  589.06  4452.1  589.27  4467.9  588.51  4473.6  586.91  4489.4  587.51
  4495.2  585.54  4511.0  586.37  4516.7  585.06  4548.3  584.62  4554.1  582.97
  4569.9  583.85  4591.5  582.89  4597.2  581.29  4628.8  581.48  4634.6  579.94
  4671.9  578.49  4715.1  572.54  4736.6  571.15  4881.9  565.15  4998.3  561.01
  4998.8  560.51  5008.6  561.01  5028.0  561.05  5111.2  561.74  5140.9  563.35
  5158.2  565.24  5201.3  574.72  5255.1  581.68  5309.0  586.44  5368.2  589.27
#Mann=5,-1,0
  4420.6     0.1       0  4881.9    0.05       0  4998.3    0.03       0
  5008.6    0.05       0  5028.0     0.1       0
Bank Sta=4998.3,5008.6
Exp/Cntr=0.3,0.1

Type RM Length L Ch R = 1,16198,382,382,382
BEGIN DESCRIPTION:
UNT 001 in BCW 29.0
END DESCRIPTION:
XS GIS Cut Line= 3
      1966264.21     13485711.25      1966675.00     13485275.00
      1967074.98     13484925.02
#Sta/Elev= 30
  4368.0  585.18  4401.4  585.29  4472.2  580.36  4521.6  578.23  4542.6  578.34
  4564.0  576.60  4677.3  573.98  4854.8  564.43  4868.3  563.95  4882.5  561.95
  4896.6  562.53  4917.7  561.35  4970.5  560.29  4988.6  558.96  4989.3  557.72
  4989.8  557.22  5000.7  557.22  5001.2  557.72  5023.7  559.77  5099.5  560.72
  5258.1  564.02  5307.5  567.16  5328.4  567.40  5385.3  570.24  5392.4  572.05
  5406.2  573.09  5428.0  578.21  5477.4  585.42  5491.6  587.02  5498.7  587.09
#Mann=5,-1,0
  4368.0     0.1       0  4854.8    0.05       0  4989.3    0.03       0
  5001.2    0.05       0  5099.5     0.1       0
Bank Sta=4989.3,5001.2
Exp/Cntr=0.3,0.1

Type RM Length L Ch R = 1,15816,482,482,482
BEGIN DESCRIPTION:
UNT 001 in BCW 28.0
END DESCRIPTION:
XS GIS Cut Line= 3
      1966420.42     13486258.17      1966971.21     13485523.04
      1967175.02     13485124.96
#Sta/Elev= 30
  4069.2  587.51  4238.6  581.47  4253.1  580.65  4267.7  578.70  4567.8  568.16
  4582.4  568.29  4617.8  565.61  4653.2  565.63  4667.8  566.68  4703.2  565.30
  4717.8  566.06  4767.8  565.28  4847.0  563.47  4865.3  561.69  4882.4  562.89
  4982.4  558.75  4990.9  556.49  4991.4  555.99  5002.8  556.49  5019.3  558.90
  5086.7  558.80  5172.5  560.91  5255.2  564.73  5287.8  567.24  5310.0  570.08
  5322.6  570.57  5337.8  574.86  5367.5  580.86  5412.5  586.74  5435.0  588.60
#Mann=5,-1,0
  4069.2     0.1       0  4865.3    0.05       0  4990.9   0.035       0
  5002.8    0.05       0  5172.5     0.1       0
Bank Sta=4990.9,5002.8
Exp/Cntr=0.3,0.1

Type RM Length L Ch R = 1,15334,597,597,597
BEGIN DESCRIPTION:
UNT 001 in BCW 27.0
END DESCRIPTION:
XS GIS Cut Line= 3
      1966835.37     13486370.99      1967375.00     13485725.00
      1967696.21     13485329.67
#Sta/Elev= 30
  4149.5  599.04  4217.5  597.90  4267.0  592.15  4281.3  588.69  4295.6  587.04
  4316.4  586.35  4324.2  584.77  4345.1  583.77  4357.5  582.07  4363.1  581.81
  4458.3  576.46  4482.6  574.14  4522.5  571.23  4607.8  566.77  4681.8  564.00
  4733.0  561.85  4870.8  558.66  4963.2  558.28  4984.1  557.54  4992.4  556.11
  4992.9  555.61  5004.4  556.11  5091.1  559.27  5162.9  563.17  5318.1  573.24
  5332.4  574.56  5361.2  579.80  5403.5  584.06  5468.0  585.37  5500.6  585.05
#Mann=11,-1,0
  4149.5     0.1       0  4357.5    0.05       0  4363.1     0.1       0
  4482.6    0.05       0  4522.5     0.1       0  4607.8    0.05       0
  4681.8     0.1       0  4733.0    0.05       0  4992.4   0.035       0
  5004.4    0.05       0  5162.9     0.1       0
Bank Sta=4992.4,5004.4
Exp/Cntr=0.3,0.1

Type RM Length L Ch R = 1,14737,103,103,103
BEGIN DESCRIPTION:
UNT 001 in BCW 26.0
END DESCRIPTION:
XS GIS Cut Line= 5
      1967147.83     13486537.68      1967703.42     13486357.11
      1967842.31     13486121.00      1967953.42     13485808.50
      1967953.42     13485559.30
#Sta/Elev= 30
  4083.0  582.31  4266.8  582.42  4553.2  567.19  4795.0  559.24  4800.8  561.03
  4816.5  559.51  4822.3  561.20  4837.9  559.11  4859.4  561.66  4875.0  559.79
  4880.8  561.80  4896.5  559.77  4912.2  560.88  4918.0  563.11  4941.1  560.40
  4947.5  556.63  4963.8  555.27  4969.1  557.85  4983.3  555.20  4983.8  554.70
  4995.3  555.20  5025.4  558.62  5081.8  557.15  5087.1  558.89  5112.7  557.76
  5169.1  559.65  5316.3  567.95  5376.3  573.30  5426.3  570.63  5522.0  571.10
#Mann=3,-1,0
  4083.0     0.1       0  4983.3    0.07       0  4995.3     0.1       0
Bank Sta=4983.3,4995.3
Exp/Cntr=0.3,0.1

Type RM Length L Ch R = 1,14634,653,653,653
BEGIN DESCRIPTION:
UNT 001 in BCW 25.0
END DESCRIPTION:
XS GIS Cut Line= 4
      1967505.49     13486653.13      1967773.73     13486431.77
      1967940.40     13486137.50      1968288.69     13485448.72
#Sta/Elev= 30
  4272.4  575.69  4298.6  575.50  4370.3  571.50  4505.1  567.13  4576.1  567.88
  4597.0  571.58  4611.3  569.64  4633.3  569.88  4649.2  566.93  4676.6  566.04
  4692.5  564.09  4823.3  558.67  4853.8  553.09  4854.3  552.59  4865.8  553.09
  4875.7  555.08  4903.8  557.17  4919.0  556.17  4978.8  557.21  5029.0  556.52
  5134.8  559.03  5262.9  566.84  5297.3  564.65  5335.4  564.05  5409.4  563.56
  5508.1  565.38  5513.7  564.35  5530.4  566.00  5641.8  571.09  5730.2  581.91
#Mann=3,-1,0
  4272.4     0.1       0  4853.8    0.07       0  4865.8     0.1       0
Bank Sta=4853.8,4865.8
Exp/Cntr=0.3,0.1

Type RM Length L Ch R = 1,13981,708,708,708
BEGIN DESCRIPTION:
UNT 001 in BCW 24.0
END DESCRIPTION:
XS GIS Cut Line= 3
      1968275.00     13486875.00      1968475.00     13486475.00
      1969224.98     13486075.01
#Sta/Elev= 30
  4551.8  576.15  4554.6  576.15  4560.2  574.13  4565.8  574.32  4588.1  570.80
  4604.9  569.46  4627.3  565.17  4632.9  565.47  4641.2  563.79  4716.7  560.54
  4730.7  560.84  4739.1  559.96  4744.7  560.68  4767.0  559.16  4850.9  557.59
  4911.4  554.96  4984.3  553.75  4984.8  553.25  4997.0  553.75  5073.0  554.84
  5133.2  554.00  5391.1  554.51  5531.7  556.10  5648.9  559.96  5695.5  567.95
  5747.0  574.71  5753.0  576.20  5797.0  581.07  5813.2  584.59  5849.0  586.82
#Mann=5,-1,0
  4551.8     0.1       0  4911.4    0.05       0  4984.3    0.03       0
  4997.0    0.05       0  5695.5     0.1       0
Bank Sta=4984.3,4997
Exp/Cntr=0.3,0.1

Type RM Length L Ch R = 1,13273,466,466,466
BEGIN DESCRIPTION:
Mapping XS 0506f0e5
END DESCRIPTION:
XS GIS Cut Line= 3
      1968684.74     13487314.73      1968968.61     13487030.86
      1969298.82     13486128.64
#Sta/Elev= 30
  4264.5  593.78  4292.8  592.25  4356.4  587.07  4377.6  584.38  4420.1  576.50
  4441.3  573.43  4483.7  570.61  4519.0  569.74  4533.2  567.78  4549.9  566.57
  4568.5  566.43  4596.8  563.46  4682.8  559.98  4938.4  552.42  4964.0  552.12
  4964.5  551.62  4976.3  551.62  4976.8  552.12  5204.6  552.78  5246.9  553.61
  5300.5  555.64  5417.6  561.34  5424.7  562.86  5485.7  568.50  5492.1  570.58
  5517.9  574.67  5572.0  581.18  5577.3  582.72  5597.2  585.04  5626.7  586.76
#Mann=5,-1,0
  4264.5     0.1       0  4549.9    0.05       0  4964.0    0.03       0
  4976.8    0.05       0  5517.9     0.1       0
Bank Sta=4964,4976.8
Exp/Cntr=0.3,0.1

Type RM Length L Ch R = 1,12807,225,225,225
BEGIN DESCRIPTION:
Mapping XS fab5f543
END DESCRIPTION:
XS GIS Cut Line= 4
      1968955.58     13487554.30      1969432.15     13487187.11
      1969541.53     13486468.36      1969759.88     13486179.81
#Sta/Elev= 30
  3940.6  578.68  3943.4  578.68  3946.9  575.88  3953.2  575.33  3961.4  572.99
  3996.7  569.04  4096.4  565.28  4175.2  560.31  4217.6  559.68  4269.4  557.00
  4395.3  554.79  4972.6  550.81  4973.1  550.31  4986.0  550.81  5110.8  553.16
  5304.2  563.69  5331.4  564.94  5373.8  568.63  5395.9  570.63  5402.2  572.11
  5410.5  572.23  5416.8  573.73  5431.3  573.87  5452.1  578.22  5460.4  578.32
  5510.4  586.11  5516.6  587.98  5537.5  590.38  5602.0  595.31  5631.1  596.16
#Mann=5,-1,0
  3940.6     0.1       0  4269.4    0.05       0  4972.6    0.03       0
  4986.0    0.05       0  5304.2     0.1       0
Bank Sta=4972.6,4986
Exp/Cntr=0.3,0.1

Type RM Length L Ch R = 1,12582,440,440,440
BEGIN DESCRIPTION:
Mapping XS 9073cba7
END DESCRIPTION:
XS GIS Cut Line= 3
      1969564.97     13488015.26      1969489.44     13487533.46
      1969851.43     13486262.59
#Sta/Elev= 30
  3754.4  595.04  3795.2  591.23  3835.6  588.71  3886.3  583.45  3906.5  580.74
  3913.6  578.64  3918.7  578.47  3957.1  570.10  3976.2  569.35  3981.3  567.82
  3987.5  567.23  4038.1  565.67  4088.7  561.81  4165.4  557.79  4302.9  554.52
  4502.6  554.10  4750.0  552.37  4885.1  550.06  4972.4  549.88  4972.9  549.38
  4985.8  549.88  5041.1  550.43  5103.5  553.08  5259.5  563.93  5270.2  565.54
  5416.4  577.35  5477.8  585.78  5484.1  587.49  5498.6  589.46  5563.5  596.75
#Mann=5,-1,0
  3754.4     0.1       0  4165.4    0.05       0  4972.4    0.03       0
  4985.8    0.05       0  5270.2     0.1       0
Bank Sta=4972.4,4985.8
Exp/Cntr=0.3,0.1

Type RM Length L Ch R = 1,12142,498,498,498
BEGIN DESCRIPTION:
UNT 001 in BCW 20.0
END DESCRIPTION:
XS GIS Cut Line= 3
      1969674.99     13488025.02      1970075.00     13487025.00
      1969975.00     13486425.03
#Sta/Elev= 30
  3889.0  595.70  3898.4  596.37  3903.8  595.69  3942.9  595.86  3957.7  594.81
  3964.4  593.02  3981.9  590.83  4006.1  590.12  4018.3  591.22  4033.1  590.57
  4082.9  586.26  4113.8  581.81  4119.2  579.57  4136.7  576.69  4148.9  573.01
  4197.3  565.02  4358.9  555.58  4449.1  552.10  4496.2  551.25  4610.6  550.52
  4711.6  551.24  4836.8  548.85  4979.6  547.80  4980.1  547.30  4993.1  547.80
  5059.8  548.96  5105.8  552.26  5358.9  560.46  5442.5  564.91  5574.3  575.49
#Mann=5,-1,0
  3889.0     0.1       0  4033.1    0.05       0  4979.6    0.03       0
  4993.1    0.05       0  5105.8     0.1       0
Bank Sta=4979.6,4993.1
Exp/Cntr=0.3,0.1

Type RM Length L Ch R = 1,11644,420,420,420
BEGIN DESCRIPTION:
UNT 001 in BCW 19.0
END DESCRIPTION:
XS GIS Cut Line= 3
      1969824.99     13487925.01      1970425.00     13487325.00
      1971088.01     13486549.54
#Sta/Elev= 30
  4160.6  582.21  4245.5  567.44  4429.3  556.36  4528.3  551.57  4669.7  547.94
  4768.7  549.06  4998.7  546.92  4999.2  546.42  5012.5  546.92  5137.0  547.67
  5143.6  548.45  5206.6  549.12  5448.8  550.63  5512.5  552.07  5682.6  552.03
  5760.6  553.66  5803.4  555.69  5817.7  555.32  5938.4  564.08  5952.7  566.32
  5959.3  568.37  5967.0  568.83  5973.5  571.37  5981.2  571.86  5987.8  574.22
  5995.5  574.38  6002.1  576.55  6016.4  576.03  6022.9  578.04  6029.4  577.82
#Mann=4,-1,0
  4160.6    0.05       0  4998.7    0.03       0  5012.5    0.05       0
  5206.6     0.1       0
Bank Sta=4998.7,5012.5
Exp/Cntr=0.3,0.1

Type RM Length L Ch R = 1,11224,467,467,467
BEGIN DESCRIPTION:
UNT 001 in BCW 18.0
END DESCRIPTION:
XS GIS Cut Line= 3
      1969925.03     13488024.99      1970525.00     13487725.00
      1971625.02     13486524.98
#Sta/Elev= 30
  4323.9  569.49  4511.1  559.04  4762.7  548.16  5023.0  545.12  5023.5  544.62
  5037.2  545.12  5122.0  550.29  5207.1  552.55  5292.2  552.12  5348.3  550.61
  5355.7  551.29  5422.7  549.41  5518.5  547.51  5716.4  548.61  5929.2  552.40
  5964.3  551.66  6084.6  555.42  6318.3  568.39  6360.8  572.75  6367.6  575.58
  6375.0  575.97  6381.8  579.20  6389.2  579.25  6396.0  582.02  6403.4  582.05
  6410.1  584.18  6438.5  587.11  6509.4  590.29  6544.6  593.01  6622.6  593.97
#Mann=4,-1,0
  4323.9    0.05       0  5023.0    0.03       0  5037.2    0.05       0
  5422.7     0.1       0
Bank Sta=5023,5037.2
Exp/Cntr=0.3,0.1

Type RM Length L Ch R = 1,10757,225,225,225
BEGIN DESCRIPTION:
UNT 001 in BCW 17.0
END DESCRIPTION:
XS GIS Cut Line= 3
      1969633.14     13489081.91      1970875.00     13487975.00
      1972084.47     13486804.19
#Sta/Elev= 30
  3312.4  584.05  3545.0  571.99  3729.8  567.09  3767.8  568.27  3927.9  569.51
  4097.9  564.37  4281.6  556.43  4550.8  550.57  4636.1  551.37  4734.8  547.75
  4990.0  545.01  5372.0  544.70  5372.5  544.20  5386.3  544.70  5580.2  545.21
  5644.7  545.77  5748.8  545.00  5785.8  545.25  5886.1  546.01  5971.2  548.38
  6113.7  551.90  6209.2  554.24  6298.0  557.92  6350.3  561.49  6435.3  576.48
  6517.7  583.60  6552.3  583.94  6581.3  587.46  6648.0  589.66  6659.3  590.12
#Mann=18,-1,0
  3312.4    0.05       0  3767.8     0.1       0  4097.9    0.05       0
  5372.0    0.04       0  5386.3    0.05       0  5580.2     0.1       0
  5644.7    0.05       0  5748.8     0.1       0  5785.8    0.05       0
  5886.1     0.1       0  5971.2    0.05       0  6113.7     0.1       0
  6209.2    0.05       0  6298.0     0.1       0  6350.3    0.05       0
  6435.3     0.1       0  6552.3    0.05       0  6648.0     0.1       0
Bank Sta=5372,5386.3
Exp/Cntr=0.3,0.1

Type RM Length L Ch R = 1,10532,670,670,670
BEGIN DESCRIPTION:
UNT 001 in BCW 16.0
END DESCRIPTION:
XS GIS Cut Line= 3
      1969938.69     13489158.30      1971153.94     13487963.88
      1972146.41     13486919.36
#Sta/Elev= 30
  3361.8  580.69  3718.1  578.60  3884.8  573.28  4040.4  565.14  4047.4  564.71
  4061.6  558.51  4082.8  558.61  4097.0  562.39  4245.4  557.15  4500.0  558.01
  4627.3  555.13  4797.0  545.06  4980.9  543.21  5143.6  545.25  5695.1  542.90
  5695.6  542.40  5709.4  542.90  5782.4  543.36  5789.8  543.29  5914.5  544.38
  6046.6  547.51  6085.0  549.20  6178.6  554.63  6232.6  561.18  6254.0  564.86
  6282.3  572.88  6310.7  578.64  6332.0  581.46  6380.2  582.54  6506.6  584.73
#Mann=13,-1,0
  3361.8     0.1       0  3718.1    0.05       0  5695.1    0.03       0
  5709.4    0.05       0  5782.4    0.08       0  5789.8     0.1       0
  5914.5    0.05       0  6046.6    0.08       0  6085.0    0.05       0
  6178.6    0.08       0  6232.6    0.05       0  6310.7    0.08       0
  6380.2    0.05       0
Bank Sta=5695.1,5709.4
Exp/Cntr=0.3,0.1

Type RM Length L Ch R = 1,9862,937,937,937
BEGIN DESCRIPTION:
UNT 001 in BCW 15.0
END DESCRIPTION:
XS GIS Cut Line= 3
      1971425.00     13489075.02      1971725.00     13487875.00
      1972174.38     13486909.18
#Sta/Elev= 30
  3806.5  575.63  3889.0  572.06  3953.4  567.73  3981.7  567.59  4084.8  563.16
  4126.1  560.08  4342.5  554.89  4476.5  548.65  4589.9  546.45  4868.2  543.83
  4901.7  542.84  4937.8  540.11  4995.0  539.67  4995.5  539.17  5009.5  539.67
  5040.9  541.18  5508.9  540.43  5639.0  543.78  5697.5  547.16  5720.4  548.88
  5737.8  551.88  5766.2  553.12  5817.4  561.54  5857.7  569.76  5886.1  573.05
  5903.5  578.04  5909.0  577.70  5914.8  579.29  6074.4  584.64  6108.7  586.10
#Mann=4,-1,0
  3806.5    0.05       0  4995.0    0.03       0  5009.5    0.05       0
  6074.4     0.1       0
Bank Sta=4995,5009.5
Exp/Cntr=0.3,0.1

Type RM Length L Ch R = 1,8925,595,595,595
BEGIN DESCRIPTION:
UNT 001 in BCW 14.0
END DESCRIPTION:
XS GIS Cut Line= 3
      1971724.98     13488825.03      1972425.00     13487625.00
      1972524.98     13487375.04
#Sta/Elev= 30
  3605.9  571.09  3613.8  570.85  3641.1  566.85  3651.0  566.36  3678.3  563.16
  3774.2  555.58  3913.1  548.82  4022.7  545.57  4212.5  542.68  4543.3  542.94
  4601.6  543.52  4709.5  542.31  4740.5  543.01  4752.5  544.32  4768.2  542.28
  4985.0  538.70  4985.5  538.20  4999.1  538.20  4999.6  538.70  5058.5  539.38
  5093.5  541.19  5112.3  544.06  5124.4  549.07  5135.2  550.43  5147.3  553.14
  5195.8  559.84  5225.4  562.24  5232.1  563.71  5249.6  565.37  5264.4  566.08
#Mann=3,-1,0
  3605.9    0.05       0  4985.0   0.035       0  4999.6    0.05       0
Bank Sta=4985,4999.6
Exp/Cntr=0.3,0.1

Type RM Length L Ch R = 1,8330,140,140,140
BEGIN DESCRIPTION:
UNT 001 in BCW 13.0
END DESCRIPTION:
XS GIS Cut Line= 3
      1971711.66     13489017.84      1972939.96     13487928.42
      1973356.19     13487070.36
#Sta/Elev= 30
  3495.4  576.44  3506.9  576.84  3542.0  575.44  3676.6  567.02  3747.7  563.59
  3782.9  560.92  3847.3  558.36  3945.9  552.13  4023.7  548.45  4186.8  543.15
  4264.6  541.74  4562.3  541.71  4774.8  540.16  4944.5  536.25  4980.5  536.90
  4994.1  536.14  4994.6  535.64  5008.7  536.14  5079.2  539.31  5093.4  540.99
  5107.6  539.33  5115.1  537.34  5121.8  541.42  5158.9  543.38  5503.1  551.46
  5615.9  552.20  5841.2  550.57  5988.2  556.04  6041.3  559.45  6090.9  561.17
#Mann=3,-1,0
  3495.4    0.05       0  4994.1   0.035       0  5008.7    0.05       0
Bank Sta=4994.1,5008.7
Exp/Cntr=0.3,0.1

Type RM Length L Ch R = 1,8190,583,583,583
BEGIN DESCRIPTION:
UNT 001 in BCW 12.0
END DESCRIPTION:
XS GIS Cut Line= 3
      1971921.77     13489003.92      1973299.77     13487797.35
      1973375.00     13487075.04
#Sta/Elev= 30
  3688.2  572.64  3725.1  571.81  3753.6  574.00  3796.3  573.76  3824.8  571.58
  3866.5  565.26  3909.2  560.31  3980.4  553.91  4058.2  549.10  4193.0  543.73
  4398.0  540.60  4419.8  541.12  4511.9  540.12  4624.8  541.16  4993.3  535.59
  4993.8  535.09  5008.0  535.59  5064.3  537.81  5114.6  541.07  5170.6  542.41
  5376.5  543.47  5503.7  545.57  5524.6  544.71  5618.1  547.11  5693.1  546.65
  5944.4  548.82  6055.0  552.19  6175.7  558.08  6205.8  560.72  6246.0  561.91
#Mann=3,-1,0
  3688.2    0.05       0  4993.3    0.03       0  5008.0    0.05       0
Bank Sta=4993.3,5008
Exp/Cntr=0.3,0.1

Type RM Length L Ch R = 1,7607,450,450,450
BEGIN DESCRIPTION:
UNT 001 in BCW 11.0
END DESCRIPTION:
XS GIS Cut Line= 3
      1972874.99     13489275.02      1973125.00     13488675.00
      1973720.29     13488080.55
#Sta/Elev= 30
  4340.3  557.74  4378.8  555.30  4431.9  552.72  4455.7  550.70  4461.1  550.68
  4508.8  547.06  4561.9  544.74  4567.8  543.94  4585.7  543.02  4676.2  539.24
  4798.0  536.10  4922.6  535.11  4975.7  534.42  4997.1  533.73  4997.6  533.23
  5011.4  533.23  5011.9  533.73  5039.8  535.09  5061.0  535.64  5117.6  538.47
  5160.0  539.58  5202.5  539.74  5280.2  538.71  5358.0  538.23  5541.9  538.31
  5570.1  539.02  5612.6  539.42  5718.6  539.51  5803.5  540.54  5831.6  540.43
#Mann=3,-1,0
  4340.3    0.05       0  4997.1    0.03       0  5011.9    0.05       0
Bank Sta=4997.1,5011.9
Exp/Cntr=0.3,0.1

Type RM Length L Ch R = 1,7157,442,442,442
BEGIN DESCRIPTION:
UNT 001 in BCW 10.0
END DESCRIPTION:
XS GIS Cut Line= 3
      1973325.00     13489625.03      1973375.00     13489025.00
      1973848.10     13488414.46
#Sta/Elev= 30
  4392.6  578.56  4412.7  577.60  4450.3  573.98  4455.4  574.04  4503.0  569.08
  4563.2  562.12  4570.7  560.84  4575.8  560.85  4663.6  552.58  4733.8  547.59
  4811.6  543.55  4924.5  535.72  4964.6  534.06  5000.8  533.28  5001.3  532.78
  5015.3  532.78  5015.8  533.28  5037.3  534.33  5072.6  534.01  5136.8  535.23
  5165.8  537.48  5180.3  537.85  5230.1  536.98  5286.2  536.79  5414.8  538.20
  5551.4  538.03  5601.3  538.62  5678.2  538.25  5736.2  539.57  5767.1  538.91
#Mann=3,-1,0
  4392.6    0.05       0  5000.8    0.03       0  5015.8    0.05       0
Bank Sta=5000.8,5015.8
Exp/Cntr=0.3,0.1

Type RM Length L Ch R = 1,6715,391,391,391
BEGIN DESCRIPTION:
UNT 001 in BCW 9.0
END DESCRIPTION:
XS GIS Cut Line= 3
      1973424.98     13489575.02      1973775.00     13489225.00
      1973978.33     13488410.09
#Sta/Elev= 30
  4477.5  571.04  4481.1  571.04  4491.7  569.43  4548.2  563.15  4576.5  559.73
  4583.6  558.50  4590.7  558.21  4619.0  555.38  4689.7  549.65  4774.5  544.83
  4816.9  541.00  4873.5  536.62  4930.1  533.83  4975.1  532.33  4988.2  531.14
  4988.7  530.64  5002.7  530.64  5003.2  531.14  5031.8  533.19  5065.3  532.77
  5096.2  533.12  5178.6  534.89  5284.6  535.50  5320.7  536.77  5367.1  536.78
  5436.3  537.71  5632.1  537.06  5692.1  537.69  5714.6  538.43  5812.4  538.84
#Mann=3,-1,0
  4477.5    0.05       0  4988.2    0.03       0  5003.2    0.05       0
Bank Sta=4988.2,5003.2
Exp/Cntr=0.3,0.1

Type RM Length L Ch R = 1,6324,38,38,38
BEGIN DESCRIPTION:
Mapping XS 465266da
END DESCRIPTION:
XS GIS Cut Line= 4
      1974039.11     13489842.34      1974146.73     13489404.89
      1974171.04     13489130.58      1973980.05     13488613.19
#Sta/Elev= 30
  4445.4  540.19  4495.2  539.18  4597.1  538.91  4744.3  536.99  4854.6  536.91
  4868.9  536.65  4915.9  534.04  4931.9  532.08  4936.9  533.01  4966.1  531.51
  4996.2  531.21  5018.8  530.20  5019.3  529.70  5033.3  529.70  5033.8  530.20
  5043.8  530.68  5048.8  532.35  5056.4  532.56  5076.5  531.71  5106.6  531.83
  5160.7  534.17  5187.9  533.52  5294.8  533.85  5380.8  534.82  5461.4  536.83
  5516.9  536.63  5571.6  537.31  5638.6  536.64  5699.5  537.93  5722.8  537.49
#Mann=3,-1,0
  4445.4    0.05       0  5018.8    0.03       0  5033.8    0.05       0
Bank Sta=5018.8,5033.8
Exp/Cntr=0.3,0.1

Type RM Length L Ch R = 1,6286,45,45,45
BEGIN DESCRIPTION:
Mapping XS 0a046c23
END DESCRIPTION:
XS GIS Cut Line= 4
      1974059.93     13489866.70      1974188.40     13489502.11
      1974198.82     13489116.70      1973983.55     13488561.16
#Sta/Elev= 30
  4411.8  539.26  4503.0  538.06  4559.6  538.30  4721.1  536.59  4798.4  536.99
  4835.5  538.97  4854.0  539.31  4905.5  538.01  4935.5  538.45  4985.5  536.98
  5005.5  537.04  5015.5  535.44  5025.6  535.22  5035.6  537.13  5055.6  536.76
  5075.6  537.63  5095.6  536.64  5115.6  537.47  5145.6  537.37  5196.5  535.49
  5202.9  533.33  5203.4  532.83  5217.4  532.83  5217.9  533.33  5344.0  534.13
  5452.9  536.62  5597.2  537.01  5627.1  536.51  5722.0  537.73  5779.7  537.49
#Mann=3,-1,0
  4411.8    0.05       0  5202.9    0.03       0  5217.9    0.05       0
Bank Sta=5202.9,5217.9
Exp/Cntr=0.3,0.1

Type RM Length L Ch R = 1,6241,116,116,116
BEGIN DESCRIPTION:
Mapping XS 3b9b096e
END DESCRIPTION:
XS GIS Cut Line= 4
      1974077.28     13489859.77      1974226.59     13489484.75
      1974250.90     13489106.28      1974007.85     13488581.98
#Sta/Elev= 30
  4411.0  538.65  4473.9  537.92  4552.1  537.91  4599.1  536.88  4665.4  536.49
  4719.3  536.49  4738.2  537.01  4834.4  536.14  4854.5  536.39  4863.6  535.52
  4934.6  531.74  4994.8  531.70  5019.3  531.16  5019.8  530.66  5033.8  530.66
  5034.3  531.16  5125.0  532.51  5155.1  533.41  5198.4  533.64  5261.4  533.15
  5318.5  534.12  5371.7  534.34  5387.2  534.60  5415.8  536.06  5461.5  536.78
  5530.2  536.47  5576.0  536.93  5644.8  536.25  5719.0  537.49  5771.8  537.51
#Mann=3,-1,0
  4411.0    0.05       0  5019.3    0.03       0  5034.3    0.05       0
Bank Sta=5019.3,5034.3
Exp/Cntr=0.3,0.1

Type RM Length L Ch R = 1,6125,632,632,632
BEGIN DESCRIPTION:
UNT 001 in BCW 8.0
END DESCRIPTION:
XS GIS Cut Line= 4
      1974101.58     13489884.09      1974290.83     13489534.23
      1974412.36     13489091.52      1973987.55     13488519.33
#Sta/Elev= 30
  4359.5  537.94  4420.1  537.15  4501.9  536.96  4574.5  535.96  4642.7  536.65
  4693.2  536.31  4715.0  536.78  4787.2  535.67  4826.8  535.86  4871.6  534.40
  4922.4  531.48  4953.5  531.24  4997.8  529.84  4998.3  529.34  5012.4  529.34
  5012.9  529.84  5014.5  530.21  5046.8  531.22  5099.0  531.51  5140.2  532.59
  5298.6  532.59  5384.1  533.59  5425.8  534.81  5540.6  536.48  5684.6  535.71
  5755.5  537.02  5790.9  537.07  5805.5  537.70  5876.5  537.81  5929.0  538.80
#Mann=3,-1,0
  4359.5    0.05       0  4997.8    0.03       0  5012.9    0.05       0
Bank Sta=4997.8,5012.9
Exp/Cntr=0.3,0.1

Type RM Length L Ch R = 1,5493,431,431,431
BEGIN DESCRIPTION:
Mapping XS 528deda1
END DESCRIPTION:
XS GIS Cut Line= 4
      1973665.69     13490002.21      1974525.03     13490054.29
      1975119.65     13489108.11      1975284.46     13488509.61
#Sta/Elev= 30
  3284.5  553.85  3624.4  540.46  3864.9  535.91  3975.1  535.85  3995.1  536.49
  4085.3  534.10  4252.7  532.89  4404.7  533.12  4487.1  535.10  4566.0  534.64
  4587.2  535.13  4602.5  534.09  4608.5  534.53  4629.7  533.91  4769.8  533.72
  4912.3  529.62  4985.4  529.80  4998.0  528.89  4998.5  528.39  5015.0  528.39
  5015.5  528.89  5030.4  529.55  5079.6  529.18  5124.9  529.94  5225.6  534.32
  5302.2  536.50  5463.2  546.10  5563.7  549.92  5711.6  552.97  5883.7  553.73
#Mann=3,-1,0
  3284.5    0.05       0  4998.0    0.03       0  5015.5    0.05       0
Bank Sta=4998,5015.5
Exp/Cntr=0.3,0.1

Type RM Length L Ch R = 1,5062,543,543,543
BEGIN DESCRIPTION:
Mapping XS 585c4bf1
END DESCRIPTION:
XS GIS Cut Line= 4
      1974919.99     13490961.37      1974811.49     13490444.92
      1975631.80     13489051.69      1975705.59     13488595.94
#Sta/Elev= 30
  3373.3  556.44  3390.0  556.42  3410.5  553.53  3441.1  545.63  3468.6  541.44
  3512.6  538.40  3584.2  537.42  3635.3  535.27  3857.3  533.23  4109.5  532.59
  4216.7  532.63  4371.0  534.27  4509.6  532.34  4655.2  533.52  4839.6  530.66
  4919.7  530.30  4990.8  526.52  4991.3  526.02  5008.5  526.52  5095.4  529.36
  5196.9  531.23  5341.3  538.00  5437.0  541.56  5516.0  543.80  5651.7  545.53
  5688.1  545.83  5737.3  547.50  5754.7  547.20  5858.9  549.59  5979.5  553.32
#Mann=5,-1,0
  3373.3    0.05       0  4990.8    0.03       0  5008.5    0.05       0
  5651.7     0.1       0  5688.1    0.05       0
Bank Sta=4990.8,5008.5
Exp/Cntr=0.3,0.1

Type RM Length L Ch R = 1,4519,550,550,550
BEGIN DESCRIPTION:
Mapping XS ac1df20b
END DESCRIPTION:
XS GIS Cut Line= 3
      1974998.14     13491000.45      1975219.48     13490510.02
      1976334.45     13489169.45
#Sta/Elev= 30
  3541.1  554.45  3566.7  553.83  3580.0  552.51  3618.5  544.66  3647.1  540.04
  3722.6  534.51  3739.6  535.77  3837.6  532.69  4100.4  530.35  4186.3  532.10
  4412.9  533.48  4505.3  531.96  4797.0  532.95  4839.9  532.55  4875.1  529.75
  4924.5  527.62  4967.5  527.29  4988.3  525.90  4993.8  524.33  4994.3  523.83
  5011.6  524.33  5017.0  525.95  5138.1  528.42  5251.3  535.26  5292.2  536.26
  5427.8  541.01  5634.1  549.86  5783.8  554.25  5821.6  556.50  5822.8  556.62
#Mann=6,-1,0
  3541.1    0.05       0  4993.8    0.03       0  5011.6    0.05       0
  5292.2     0.1       0  5427.8    0.05       0  5821.6     0.1       0
Bank Sta=4993.8,5011.6
Exp/Cntr=0.3,0.1

Type RM Length L Ch R = 1,3969,313,313,313
BEGIN DESCRIPTION:
Mapping XS ea547250
END DESCRIPTION:
XS GIS Cut Line= 5
      1974976.45     13491048.19      1975523.30     13490531.72
      1975783.71     13490271.31      1976426.08     13489993.53
      1977146.54     13489906.73
#Sta/Elev= 30
  3820.1  553.31  3892.0  552.57  3962.8  538.91  4245.6  529.99  4917.7  531.73
  4931.8  531.44  4959.9  523.39  4960.4  522.89  4978.3  523.39  5021.6  524.46
  5039.6  528.68  5068.6  527.49  5074.0  529.31  5092.0  527.27  5097.5  529.71
  5115.5  527.24  5121.0  530.28  5144.5  527.02  5149.9  529.30  5183.9  529.16
  5236.1  531.68  5301.8  528.92  5343.3  535.03  5419.2  536.95  5500.6  532.86
  5587.1  531.96  5754.3  534.13  6005.7  542.12  6243.7  553.37  6366.1  555.03
#Mann=5,-1,0
  3820.1    0.05       0  4959.9    0.03       0  4978.3    0.05       0
  5183.9     0.1       0  5587.1    0.05       0
Bank Sta=4959.9,4978.3
Exp/Cntr=0.3,0.1

Type RM Length L Ch R = 1,3656,368,368,368
BEGIN DESCRIPTION:
UNT 001 in BCW 6.0
END DESCRIPTION:
XS GIS Cut Line= 4
      1974924.99     13491525.02      1975514.62     13490727.04
      1976356.63     13490301.69      1976855.75     13490158.46
#Sta/Elev= 30
  3379.5  566.82  3487.1  564.89  3528.7  562.19  3629.0  558.52  3672.9  553.53
  3693.7  547.69  3708.3  545.53  3778.4  543.86  3808.6  543.01  3829.4  540.11
  4138.0  529.69  4432.7  529.11  4767.1  530.86  4980.8  523.33  4981.3  522.83
  4999.3  523.33  5101.5  524.36  5212.9  532.77  5302.1  537.72  5470.4  538.78
  5576.8  541.07  5649.5  544.87  5716.9  550.31  5722.1  549.83  5755.9  555.05
  5761.1  554.03  5789.6  559.97  5794.8  558.85  5802.3  561.59  5834.3  567.35
#Mann=4,-1,0
  3379.5     0.1       0  3778.4    0.05       0  4980.8    0.03       0
  4999.3    0.05       0
Bank Sta=4980.8,4999.3
Exp/Cntr=0.3,0.1

Type RM Length L Ch R = 1,3288,458,458,458
BEGIN DESCRIPTION:
UNT 001 in BCW 5.0
END DESCRIPTION:
XS GIS Cut Line= 3
      1974998.16     13491712.25      1976225.00     13490775.00
      1976824.98     13490225.02
#Sta/Elev= 30
  3454.7  555.72  3472.2  553.90  3478.5  554.38  3507.6  551.86  3533.3  550.79
  3684.2  544.15  3762.5  541.20  3885.8  536.07  3950.2  534.22  4099.8  530.40
  4256.1  528.01  4527.9  527.60  4663.0  528.78  4777.3  526.93  4841.7  524.51
  4948.3  524.67  5010.6  523.22  5011.1  522.72  5029.1  523.22  5125.9  526.79
  5211.0  532.92  5331.3  536.80  5394.8  537.68  5642.7  548.08  5692.0  551.12
  5756.1  557.36  5762.9  557.11  5770.3  558.85  5777.1  558.68  5812.5  561.64
#Mann=6,-1,0
  3454.7     0.1       0  3533.3    0.05       0  3684.2     0.1       0
  3762.5    0.05       0  5010.6    0.03       0  5029.1    0.05       0
Bank Sta=5010.6,5029.1
Exp/Cntr=0.3,0.1

Type RM Length L Ch R = 1,2830,468,468,468
BEGIN DESCRIPTION:
UNT 001 in BCW 4.0
END DESCRIPTION:
XS GIS Cut Line= 3
      1975224.98     13492025.01      1976225.00     13491225.00
      1977424.99     13491325.00
#Sta/Elev= 30
  3703.5  575.99  3753.9  573.93  3810.0  560.42  3858.2  553.81  3888.4  549.59
  3964.7  544.49  3981.3  543.95  3987.7  545.32  4030.9  541.47  4045.3  538.31
  4158.9  533.68  4279.8  532.86  4301.4  527.85  4379.9  524.95  4535.9  522.78
  4656.8  524.98  4813.7  522.18  4995.0  521.83  4995.5  521.33  5013.5  521.83
  5204.9  531.07  5265.1  532.20  5465.8  528.83  5556.1  529.10  5576.2  530.64
  5616.3  529.16  5786.9  530.17  6007.1  538.89  6104.7  542.87  6188.3  544.79
#Mann=7,-1,0
  3703.5     0.1       0  3858.2    0.05       0  3964.7     0.1       0
  4995.0    0.07       0  5013.5     0.1       0  6007.1    0.05       0
  6104.7     0.1       0
Bank Sta=4995,5013.5
Exp/Cntr=0.3,0.1
