--- UNT 033 in BCW.prj (project) ---

Proj Title=UNT 033 in BCW Base Level Engineering
Current Plan=p02
Default Exp/Contr=0.3,0.1
English Units
Geom File=g01
Flow File=f01
Plan File=p02
Y Axis Title=Elevation
X Axis Title(PF)=Main Channel Distance
X Axis Title(XS)=Station
BEGIN DESCRIPTION:
UNT 033 in BCW
END DESCRIPTION:
DSS Export Rating Curves= 0
DSS Export Rating Curve Sorted= 0
DSS Export Volume Flow Curves= 0
DXF OffsetX= 0
DXF OffsetY= 0
DXF ScaleX= 1
DXF ScaleY= 10

--- UNT 033 in BCW.p02 (plan) ---

Plan Title=Multiple Run
Program Version=5.07
Short Identifier=Multiple Run
Geom File=g01
Flow File=f01
Subcritical Flow
K Sum by GR= 0
Std Step Tol= 0.01
Critical Tol= 0.01
Num of Std Step Trials= 20
Max Error Tol= 0.3
Flow Tol Ratio= 0.001
Split Flow NTrial= 30
Split Flow Tol= 0.02
Split Flow Ratio= 0.02
Log Output Level= 0
Friction Slope Method= 1
Unsteady Friction Slope Method= 2
Unsteady Bridges Friction Slope Method= 1
Parabolic Critical Depth
Global Vel Dist= 1 , 1 , 1
Global Log Level= 0
CheckData=True
Encroach Param=-1 ,0,0, 0
BEGIN DESCRIPTION:
Multiple Run
END DESCRIPTION:
Computation Interval=1MIN
Output Interval=1HOUR
Instantaneous Interval=1HOUR
Mapping Interval=1HOUR
Computation Time Step Use Courant=        0
Computation Time Step Use Time Series=    0
Computation Time Step Count To Double=0
Computation Time Step Max Doubling=0
Computation Time Step Max Halving=0
Computation Time Step Residence Courant=0
Run HTab= 0
Run UNet= 0
Run Sediment= 0
Run PostProcess= 0
Run WQNet= 0
Run RASMapper= 0
UNET Theta= 1
UNET Theta Warmup= 1
UNET ZTol= 0.02
UNET ZSATol= 0.02
UNET MxIter= 20
UNET Max Iter WO Improvement= 0
UNET MaxInSteps= 0
UNET DtIC= 0
UNET DtMin= 0
UNET MaxCRTS= 20
UNET WFStab= 2
UNET SFStab= 1
UNET WFX= 1
UNET SFX= 1
UNET 1D Methodology=Finite Difference
UNET DSS MLevel= 4
UNET Pardiso=0
UNET DZMax Abort= 100
UNET Use Existing IB Tables=-1
UNET Froude Reduction=False
UNET Froude Limit= 0.8
UNET Froude Power= 4
UNET D1 Cores= 0
UNET D2 Coriolis=0
UNET D2 Cores= 0
UNET D2 Theta= 1
UNET D2 Theta Warmup= 1
UNET D2 Z Tol= 0.01
UNET D2 Volume Tol= 0.01
UNET D2 Max Iterations= 20
UNET D2 Equation= 0
UNET D2 RampUpFraction=0.1
UNET D2 TimeSlices= 1
UNET D2 BCVolumeCheck=0
UNET D1D2 MaxIter= 0
UNET D1D2 ZTol=0.01
UNET D1D2 QTol=0.1
UNET D1D2 MinQTol=1
Write IC File= 0
Write IC File at Fixed DateTime=0
Write IC File at Sim End=0
Echo Input=False
Echo Parameters=False
Echo Output=False
Write Detailed= 0
HDF Write Warmup=0
HDF Write Time Slices=0
HDF Flush=0
HDF Face Node Velocities=0
HDF Compression= 1
HDF Chunk Size= 1
HDF Spatial Parts= 1
HDF Use Max Rows=0
HDF Fixed Rows= 1
Calibration Method= 0
Calibration Iterations= 20
Calibration Max Change=0.05
Calibration Tolerance=0.2
Calibration Maximum=1.5
Calibration Minimum=0.5
Calibration Optimization Method= 1
WQ AD Non Conservative
WQ ULTIMATE=-1
WQ Max Comp Step=1HOUR
WQ Output Interval=15MIN
WQ Output Selected Increments= 0
WQ Output face flow=0
WQ Output face velocity=0
WQ Output face area=0
WQ Output face dispersion=0
WQ Output cell volume=0
WQ Output cell surface area=0
WQ Output cell continuity=0
WQ Output cumulative cell continuity=0
WQ Output face conc=0
WQ Output face dconc_dx=0
WQ Output face courant=0
WQ Output face peclet=0
WQ Output face adv mass=0
WQ Output face disp mass=0
WQ Output cell mass=0
WQ Output cell source sink temp=0
WQ Output nsm pathways=0
WQ Output nsm derived pathways=0
WQ Output MaxMinRange=-1
WQ Daily Max Min Mean=-1
WQ Daily Range=0
WQ Daily Time=0
WQ Create Restart=0
WQ Fixed Restart=0
WQ System Summary=0
WQ Write To DSS=0
WQ Use Fixed Temperature=0
Sorting and Armoring Iterations= 10
XS Update Threshold= 0.02
Bed Roughness Predictor= 0
Hydraulics Update Threshold= 0.02
Energy Slope Method= 1
Volume Change Method= 1
Sediment Retention Method= 0
XS Weighting Method= 0
Number of US Weighted Cross Sections= 1
Number of DS Weighted Cross Sections= 1
Upstream XS Weight=0
Main XS Weight=1
Downstream XS Weight=0
Number of DS XS's Weighted with US Boundary= 1
Upstream Boundary Weight= 1
Weight of XSs Associated with US Boundary= 0
Number of US XS's Weighted with DS Boundary= 1
Downstream Boundary Weight= 0.5
Weight of XSs Associated with DS Boundary= 0.5
Percentile Method= 0
Sediment Output Level= 3
Mass or Volume Output= 0
Output Increment Type= 1
Profile and TS Output Increment= 1
XS Output Flag= 0
XS Output Increment= 10
Write Gradation File= 0
Read Gradation Hotstart= 0
Write HDF5 File= 1
Write Binary Output= 1
Write DSS Sediment File= 0
SV Curve= 0
Specific Gage Flag= 0

--- UNT 033 in BCW.f01 (steady flow) ---

Flow Title=Multiple
Program Version=5.05
Number of Profiles= 7
Profile Names=10-year,25-year,50-year,1pct_min,100-year,1pct_plu,500-year
River Rch & RM=UNT 033 in BCW,Reach-1         ,29592
     708    1012    1269     786    1569    3131    2402
River Rch & RM=UNT 033 in BCW,Reach-1         ,28421
     854    1234    1557     970    1935    3861    2997
River Rch & RM=UNT 033 in BCW,Reach-1         ,25604
    1166    1707    2175    1365    2724    5436    4288
River Rch & RM=UNT 033 in BCW,Reach-1         ,19106
    1492    2209    2833    1790    3571    7124    5690
River Rch & RM=UNT 033 in BCW,Reach-1         ,13063
    1564    2320    2979    1883    3758    7498    6001
River Rch & RM=UNT 033 in BCW,Reach-1         ,12548
    1881    2804    3612    2290    4568    9115    7337
Boundary for River Rch & Prof#=UNT 033 in BCW,Reach-1         , 1
Up Type= 0
Dn Type= 3
Dn Slope=0.005
Boundary for River Rch & Prof#=UNT 033 in BCW,Reach-1         , 2
Up Type= 0
Dn Type= 3
Dn Slope=0.005
Boundary for River Rch & Prof#=UNT 033 in BCW,Reach-1         , 3
Up Type= 0
Dn Type= 3
Dn Slope=0.005
Boundary for River Rch & Prof#=UNT 033 in BCW,Reach-1         , 4
Up Type= 0
Dn Type= 3
Dn Slope=0.005
Boundary for River Rch & Prof#=UNT 033 in BCW,Reach-1         , 5
Up Type= 0
Dn Type= 3
Dn Slope=0.005
Boundary for River Rch & Prof#=UNT 033 in BCW,Reach-1         , 6
Up Type= 0
Dn Type= 3
Dn Slope=0.005
Boundary for River Rch & Prof#=UNT 033 in BCW,Reach-1         , 7
Up Type= 0
Dn Type= 3
Dn Slope=0.005
DSS Import GetInterval= 0
DSS Import GetPeak= 0
DSS Import FillOption= 0

--- UNT 033 in BCW.g01 (geometry) ---

Geom Title=Existing Conditions
Program Version=5.05

River Reach=UNT 033 in BCW  ,Reach-1
Reach XY= 30
      1959032.99     13563976.38      1959624.57     13564544.11
       1960160.6     13564597.93       1961330.8     13564194.54
       1962700.8     13562824.54       1963590.8     13562854.54
      1964094.55     13562179.36       1965140.8     13562424.54
       1965565.9     13561838.65       1966440.8     13561494.54
      1966989.03     13560511.69      1967786.26     13560290.86
       1968120.8     13560554.54      1969015.18     13560561.29
      1968908.57     13559339.05      1969274.51     13558543.06
      1968985.88     13557937.59       1969440.8     13557204.54
       1969270.8     13556604.54      1969525.11     13555758.92
       1971240.8     13554804.54       1971770.8     13554134.54
       1971700.8     13553754.54       1972400.8     13553554.54
       1972920.8     13552784.54       1973570.8     13552544.54
       1974130.8     13551644.54       1973810.8     13550434.54
       1973130.8     13549884.54       1972940.8     13548644.54

Type RM Length L Ch R = 1 ,29592   ,479,479,479
BEGIN DESCRIPTION:
UNT 033 in BCW 23.0
END DESCRIPTION:
XS GIS Cut Line= 3
      1958926.62     13564876.29       1959213.1     13564162.71
      1959174.04     13563490.88
#Sta/Elev= 30
  4219.8  713.59  4305.7  709.93    4372  704.74    4580  696.22  4619.9  693.53
  4901.3  690.26  4962.4  689.21  4984.8  686.87  5002.1  686.81  5036.5   687.7
  5043.8  686.34  5044.3  685.54  5049.8  686.34  5089.7  687.93  5104.1  688.43
  5156.7  689.55    5203  692.66  5256.9  693.97  5301.9  701.09    5327  703.09
  5424.9   704.4  5487.3  705.15  5507.3  703.82  5517.3  704.45  5537.4  709.16
  5547.4  709.92  5597.5  710.24  5617.5  712.85  5657.1  722.44  5661.7  722.44
#Mann= 11 ,-1 , 0
  4219.8      .1       0  4901.3     .12       0  4962.4     .16       0
  5002.1      .1       0  5043.8     .07       0  5049.8      .1       0
  5089.7     .16       0  5104.1      .1       0    5203     .05       0
  5301.9     .08       0  5424.9      .1       0
Bank Sta=5043.8,5049.8
XS Rating Curve= 0 ,0
Exp/Cntr=0.3,0.1

Type RM Length L Ch R = 1 ,29113   ,251,251,251
BEGIN DESCRIPTION:
UNT 033 in BCW 22.0
END DESCRIPTION:
XS GIS Cut Line= 3
      1959273.01     13565066.33      1959627.16     13564324.17
      1959444.87     13563470.03
#Sta/Elev= 30
    4363  701.61  4748.7  692.05    4852  690.85  4884.9  689.63  4934.8  685.22
  5029.1   684.4  5029.6   683.6  5035.1   684.4  5253.4  686.98  5330.4  690.14
  5354.9  690.26  5378.8  690.93  5429.9  696.92    5481  697.75  5521.9  695.97
  5542.5  697.53  5583.3   699.3  5655.4  697.61  5685.5  700.77  5716.2  701.79
  5767.3  700.73  5793.7  705.34  5818.4  706.69  5900.2  718.42  5963.7  722.42
  6022.9   725.4  6031.1  723.36  6036.2  726.09  6043.4  723.66  6058.7  723.69
#Mann= 9 ,-1 , 0
    4363      .1       0  4934.8     .16       0  5029.1     .07       0
  5035.1     .16       0  5253.4     .08       0  5330.4     .05       0
  5354.9     .08       0  5542.5      .1       0  5963.7     .05       0
Bank Sta=5029.1,5035.1
XS Rating Curve= 0 ,0
Exp/Cntr=0.3,0.1

Type RM Length L Ch R = 1 ,28862   ,441,441,441
BEGIN DESCRIPTION:
Mapping XS 1cf9ff7d
END DESCRIPTION:
XS GIS Cut Line= 3
      1960202.68      13565214.8      1959647.99     13564308.55
      1959484.11      13563619.2
#Sta/Elev= 30
  4173.1  713.91  4294.6  707.88  4484.1  691.71  4578.9  688.04  4700.9  685.26
  4941.7  682.87  5003.5  682.44    5004  681.64  5009.5  682.44  5030.2  683.22
  5076.7  683.53  5287.3   687.1  5342.1  689.84  5404.4  690.96  5441.4  696.42
  5496.3  697.55  5547.6  695.89    5567  697.31    5599  699.07  5629.9  699.03
  5681.3  697.14  5699.6  699.45  5704.8  698.65  5712.1  700.18  5753.2  701.54
  5794.3  699.92  5825.2  704.18  5866.3  707.42  5915.6  715.42  5944.2   718.2
#Mann= 8 ,-1 , 0
  4173.1      .1       0  4941.7     .16       0  5003.5     .07       0
  5009.5     .16       0  5030.2      .1       0  5076.7     .16       0
  5287.3     .08       0    5567      .1       0
Bank Sta=5003.5,5009.5
XS Rating Curve= 0 ,0
Exp/Cntr=0.3,0.1

Type RM Length L Ch R = 1 ,28421   ,464,464,464
BEGIN DESCRIPTION:
Mapping XS be6b516b
END DESCRIPTION:
XS GIS Cut Line= 4
      1960595.91     13565324.16      1960687.05     13564938.75
      1959666.22     13564300.73      1959481.31     13563514.23
#Sta/Elev= 30
  3960.9  709.59  4329.4  694.26  4507.8     692  4621.5  691.85  4731.4  692.74
  4795.7  686.34  4859.6  684.45  4962.8  682.47  4974.8  680.73  4975.3  679.93
  4980.9  680.73  5055.5  682.12  5076.5  682.08  5190.3  682.13  5251.4  682.49
    5304  682.64  5447.3  684.57  5531.5  685.58  5603.7  687.13  5689.9  690.01
  5751.6   696.1  5868.8   696.8  5976.8  696.42  6049.5  700.65  6100.8  698.27
  6215.7  711.69  6221.2  712.64  6317.7  721.23  6347.4  723.04  6368.7  719.96
#Mann= 20 ,-1 , 0
  3960.9      .1       0  4329.4     .08       0  4507.8     .05       0
  4621.5      .1       0  4859.6     .05       0  4962.8      .1       0
  4974.8     .07       0  4980.9      .1       0  5055.5     .08       0
  5076.5     .05       0  5190.3     .16       0  5251.4     .05       0
    5304     .16       0  5447.3     .05       0  5531.5     .16       0
  5603.7     .08       0  5868.8      .1       0  6215.7     .05       0
  6221.2      .1       0  6317.7     .05       0
Bank Sta=4974.8,4980.9
XS Rating Curve= 0 ,0
Exp/Cntr=0.3,0.1

Type RM Length L Ch R = 1 ,27957   ,339,339,339
BEGIN DESCRIPTION:
UNT 033 in BCW 20.0
END DESCRIPTION:
XS GIS Cut Line= 4
        1961075.     13565275.01      1960889.31     13564637.02
      1959789.05     13563907.85      1959619.91     13563560.89
#Sta/Elev= 30
  3945.6  731.48  3995.9  720.17  4001.1  722.14  4033.9  711.08  4137.5  705.12
  4268.1  702.83    4552   693.9  4643.1  687.83  4879.7  684.41  4967.9   684.1
    4989  682.19    4995  677.69  4995.5  676.89  5001.1  677.69  5025.1  681.23
  5067.1   680.3  5105.4  680.24  5254.5  680.33  5336.6  681.25  5452.2  682.29
  5567.7  683.61  5629.3  684.84  5683.3  685.48  5798.9  687.61  6000.9  691.66
  6112.5  697.43  6181.2  700.87  6196.8  706.95  6203.7  705.17    6316  713.86
#Mann= 20 ,-1 , 0
  3945.6      .1       0  4033.9     .05       0  4137.5     .08       0
  4268.1      .1       0    4552     .05       0  4643.1      .1       0
  4879.7     .05       0    4995     .07       0  5001.1      .1       0
  5067.1     .05       0  5105.4     .08       0  5254.5     .05       0
  5336.6     .08       0  5452.2     .08       0  5567.7      .1       0
  5629.3     .05       0  5683.3     .08       0  5798.9      .1       0
  6112.5      .1       0  6196.8     .05       0
Bank Sta=4995,5001.1
XS Rating Curve= 0 ,0
Exp/Cntr=0.3,0.1

Type RM Length L Ch R = 1 ,27618   ,400,400,400
BEGIN DESCRIPTION:
UNT 033 in BCW 19.0
END DESCRIPTION:
XS GIS Cut Line= 3
      1961353.73     13564934.35        1960825.       13564225.
      1960190.53     13563445.62
#Sta/Elev= 30
  4139.3  705.92  4155.5  705.59  4177.9  705.14  4230.6  703.91  4245.2  701.35
  4280.7  700.89  4295.3  698.93  4380.8  697.05  4395.4  694.68  4530.9   687.3
  4574.7   683.5    4631  682.08  4745.7  675.81  4821.4  674.68  4821.9  673.88
  4827.6  674.68  4834.7  674.78  4884.9  674.75  5194.2  676.14  5350.8  678.93
    5707  689.87  5742.2  692.44  5862.2  696.04  5913.1  701.34  5926.6  701.04
  5954.8  694.48  5969.1   694.2  5983.5  695.38  6004.3  700.92    6029  701.99
#Mann= 7 ,-1 , 0
  4139.3     .08       0  4155.5     .05       0  4177.9      .1       0
  4821.4     .07       0  4827.6      .1       0  4834.7     .12       0
  4884.9      .1       0
Bank Sta=4821.4,4827.6
XS Rating Curve= 0 ,0
Exp/Cntr=0.3,0.1

Type RM Length L Ch R = 1 ,27218   ,362,362,362
BEGIN DESCRIPTION:
UNT 033 in BCW 18.0
END DESCRIPTION:
XS GIS Cut Line= 3
      1961466.58     13564669.59        1961175.       13564075.
      1960825.03     13563675.03
#Sta/Elev= 30
  4470.9  686.14  4596.2  680.94  4631.9  680.49  4663.7  679.08  4669.2  679.25
  4676.5  678.71  4714.2  677.82  4736.3  676.66  4753.6  675.09  4787.9  675.18
  4854.7  673.67  4954.9  672.81  5057.2  672.86  5076.6  672.45  5077.1  671.65
  5082.3  671.65  5082.8  672.45  5168.7  672.66  5274.3  673.57  5367.1  674.98
  5494.3  678.86    5537   681.4  5551.2  681.32  5572.1  682.21  5600.6  684.26
  5608.2  685.44  5629.1  686.77  5636.6  687.92  5650.9  689.29  5664.6  690.03
#Mann= 5 ,-1 , 0
  4470.9      .1       0  4736.3     .12       0  5076.6     .07       0
  5082.8     .12       0  5274.3      .1       0
Bank Sta=5076.6,5082.8
XS Rating Curve= 0 ,0
Exp/Cntr=0.3,0.1

Type RM Length L Ch R = 1 ,26856   ,153,153,153
BEGIN DESCRIPTION:
UNT 033 in BCW 17.0
END DESCRIPTION:
XS GIS Cut Line= 3
      1961887.58     13564765.08       1961631.5     13564131.38
       1960985.6     13563429.13
#Sta/Elev= 30
  4148.4   698.9  4196.2  700.42  4472.1   684.2  4700.9  677.96    4807  673.21
  4862.3   669.7  4911.6  668.98  4947.4  665.91  4954.2  667.03  4975.7   664.6
  4996.7  665.63  5007.8  663.53  5008.3  662.73    5014  663.53  5039.2  664.08
    5046  665.73  5053.4  664.65  5060.2  666.68  5067.6  665.64  5074.4  668.05
  5081.8  667.02  5088.6  668.67  5095.9  667.79  5131.1  670.48  5180.4  670.89
    5223  669.16  5362.6  672.27    5591  679.82  5718.7  688.77    5786  691.43
#Mann= 6 ,-1 , 0
  4148.4      .1       0  4700.9     .12       0    4807     .05       0
  5007.8    .033       0    5014     .05       0  5362.6      .1       0
Bank Sta=5007.8,5014
XS Rating Curve= 0 ,0
Exp/Cntr=0.3,0.1

Type RM Length L Ch R = 1 ,26703   ,123,123,123
BEGIN DESCRIPTION:
UNT 033 in BCW 16.0
END DESCRIPTION:
XS GIS Cut Line= 3
      1962180.09       13564581.       1961672.3     13563953.42
      1961169.83     13563362.44
#Sta/Elev= 30
    4123  689.76    4557  681.31  4593.7  678.08  4600.2  680.31  4614.5  677.41
  4635.4  679.66  4735.3  672.25  4783.8  671.49  4870.4   674.4  4977.1  671.45
  5069.4  671.54    5076  674.04    5098  671.52  5104.5  674.01  5161.7  671.18
  5182.5  673.08  5211.1  670.97  5373.4  671.09  5427.6  669.59  5428.1  668.79
  5433.8  669.59  5516.4  672.28  5551.5  676.69  5565.8  674.29  5600.9  678.07
  5608.7  676.68  5629.5  681.01  5643.8  679.34  5678.9  685.93    5706   687.3
#Mann= 5 ,-1 , 0
    4123      .1       0  4783.8     .05       0  5373.4      .1       0
  5427.6    .033       0  5433.8      .1       0
Bank Sta=5427.6,5433.8
XS Rating Curve= 0 ,0
Exp/Cntr=0.3,0.1

Type RM Length L Ch R = 1 ,26580   ,399,399,399
BEGIN DESCRIPTION:
UNT 033 in BCW 15.0
END DESCRIPTION:
XS GIS Cut Line= 3
      1962284.27     13564471.64      1961779.07     13563901.34
      1961303.34     13563248.84
#Sta/Elev= 30
  4131.1  684.97  4190.5  683.92    4309  680.57  4333.7  679.85  4579.9  672.59
  4609.6  669.24  4620.2  669.52  4715.4  666.71  4763.4   665.4  4815.4  663.96
  4850.9  664.83  4908.2  664.39    4979  664.72  5103.9   663.9  5215.2  663.88
  5228.8  662.62  5272.1  662.37    5280  663.73  5300.9  662.85  5306.1  660.95
  5306.6  660.15  5312.3  660.95  5353.6  666.37  5388.3  666.34  5408.2  665.89
  5478.5  669.54  5487.1  668.96  5548.4  674.92  5603.3  677.42  5700.5  683.81
#Mann= 20 ,-1 , 0
  4131.1     .08       0  4190.5     .05       0    4309      .1       0
  4333.7     .05       0  4579.9      .1       0  4620.2     .05       0
  4715.4      .1       0  4763.4     .05       0  4850.9      .1       0
  4908.2     .05       0    4979     .08       0  5103.9     .05       0
  5228.8     .05       0  5306.1     .07       0  5312.3     .05       0
  5353.6      .1       0  5388.3     .08       0  5478.5      .1       0
  5548.4     .08       0  5603.3      .1       0
Bank Sta=5306.1,5312.3
XS Rating Curve= 0 ,0
Exp/Cntr=0.3,0.1

Type RM Length L Ch R = 1 ,26181   ,577,577,577
BEGIN DESCRIPTION:
Mapping XS aac58b26
END DESCRIPTION:
XS GIS Cut Line= 4
      1962296.25     13564343.75      1962228.55     13563828.16
      1961848.34     13563416.71      1961270.17      13563171.9
#Sta/Elev= 30
    4056  682.59  4145.5   680.7  4296.8  675.97  4306.9  676.13  4616.2  665.67
  4750.6  663.72  4870.8  664.13  4892.4  664.78  4920.7  663.99  5058.7   663.5
  5059.2   662.7  5064.5   662.7    5065   663.5  5108.6  663.98  5231.3  664.66
  5330.6  666.48  5360.5  666.56  5513.5  670.97  5519.9  672.06  5566.3  673.86
  5584.6  675.45    5590  675.13  5613.7  677.98  5619.1  677.61  5637.3  679.93
    5661  681.57  5666.5   681.2  5713.8  684.33  5759.5  685.27  5764.1  685.27
#Mann= 6 ,-1 , 0
    4056      .1       0  5058.7     .07       0    5065      .1       0
  5108.6     .12       0  5330.6      .1       0  5759.5     .05       0
Bank Sta=5058.7,5065
XS Rating Curve= 0 ,0
Exp/Cntr=0.3,0.1

Type RM Length L Ch R = 1 ,25604   ,462,462,462
BEGIN DESCRIPTION:
UNT 033 in BCW 14.0
END DESCRIPTION:
XS GIS Cut Line= 3
        1962375.     13563975.02        1962275.       13563175.
      1961975.02     13562375.04
#Sta/Elev= 30
  4171.9  677.24  4222.3  674.29  4272.7  672.44  4383.6  666.39  4451.6  664.17
  4514.6  662.71  4585.1  663.09  4612.8   662.4    4695  661.83    4706  662.35
  4779.1     662  4995.2  658.98  5006.8  658.72  5007.3  657.92  5013.1  657.92
  5013.6  658.72  5031.5  659.36  5053.8  658.88  5084.9  659.85  5194.4  661.22
    5384  662.24  5426.7  663.36  5469.4  663.13  5608.3   665.6  5707.1  668.66
  5725.7  670.03    5732   671.1  5737.3     671  5768.5  673.43  5832.5  676.16
#Mann= 5 ,-1 , 0
  4171.9      .1       0    4695     .05       0  4995.2      .1       0
  5006.8     .07       0  5013.6      .1       0
Bank Sta=5006.8,5013.6
XS Rating Curve= 0 ,0
Exp/Cntr=0.3,0.1

Type RM Length L Ch R = 1 ,25142   ,595,595,595
BEGIN DESCRIPTION:
UNT 033 in BCW 13.0
END DESCRIPTION:
XS GIS Cut Line= 3
       1962895.2      13563687.5        1962625.       13562925.
      1962181.66     13562286.48
#Sta/Elev= 30
  4180.5  664.61  4246.8  663.28  4284.9  660.99  4315.8  660.12  4346.7  660.48
  4372.3   659.2    4434  658.44  4732.3  657.65    4794   658.2  4921.5  656.09
  4964.8  655.09  4965.3  654.29  4971.1  654.29  4971.6  655.09  4979.3  655.81
    5003  655.39    5026  656.57  5038.8  655.75  5054.2  656.47  5277.2   658.8
    5306  659.83  5327.8  659.55  5506.8  665.83  5527.7  667.35  5578.4  668.78
  5608.1  670.55  5614.2  670.17  5715.5  673.46  5736.4  673.28  5766.8  675.03
#Mann= 5 ,-1 , 0
  4180.5      .1       0  4921.5     .12       0  4964.8     .07       0
  4971.6     .12       0  5054.2      .1       0
Bank Sta=4964.8,4971.6
XS Rating Curve= 0 ,0
Exp/Cntr=0.3,0.1

Type RM Length L Ch R = 1 ,24547   ,452,452,452
BEGIN DESCRIPTION:
Mapping XS e5953771
END DESCRIPTION:
XS GIS Cut Line= 3
      1963381.36     13563931.55      1963129.63     13562751.04
      1962709.56     13562170.66
#Sta/Elev= 30
  3827.2  666.73  4118.3  658.98  4261.8  657.24  4355.4  654.82  4590.5  653.13
  4682.6   653.7  4883.8  652.65  4979.1   651.7  4996.1  649.56  4996.6  648.76
  5002.5  648.76    5003  649.56    5020  651.68  5032.3   651.8  5070.2  652.11
  5091.1  653.29  5099.6  652.53  5191.6  653.64  5321.5  658.33    5579  664.82
  5614.6  664.61    5644   666.3  5650.2  665.67  5658.7  666.42  5664.9  665.07
  5671.3  665.88  5700.5  665.45  5708.3  666.26  5721.3  664.82  5750.7  665.57
#Mann= 5 ,-1 , 0
  3827.2      .1       0  4883.8     .12       0  4996.1     .07       0
    5003     .12       0  5032.3      .1       0
Bank Sta=4996.1,5003
XS Rating Curve= 0 ,0
Exp/Cntr=0.3,0.1

Type RM Length L Ch R = 1 ,24095   ,594,594,594
BEGIN DESCRIPTION:
Mapping XS 623f592f
END DESCRIPTION:
XS GIS Cut Line= 3
      1963889.18     13564209.35      1963481.15     13562646.74
      1963199.68     13561940.89
#Sta/Elev= 30
  3610.1  665.92  3955.7  661.18  4002.4  659.92  4083.3  659.52  4118.6  658.19
  4123.8  658.81  4204.7   656.9  4255.4  654.91  4296.7  654.02  4320.9   654.4
  4437.1  651.44  4586.1   650.5    4791  651.29  4978.9  650.13  4991.9  649.12
  5006.4  648.47  5006.9  647.67  5012.8  647.67  5013.3  648.47  5061.5   650.4
  5109.5  649.73  5192.4  650.12  5230.3     650  5323.9  651.39  5463.8  654.66
  5685.8  663.78  5829.9  670.49  5871.8  671.48  5901.5  673.67    5985  677.03
#Mann= 5 ,-1 , 0
  3610.1      .1       0  4991.9     .12       0  5006.4     .07       0
  5013.3     .12       0  5192.4      .1       0
Bank Sta=5006.4,5013.3
XS Rating Curve= 0 ,0
Exp/Cntr=0.3,0.1

Type RM Length L Ch R = 1 ,23501   ,65,65,65
BEGIN DESCRIPTION:
Mapping XS 5b3137c3
END DESCRIPTION:
XS GIS Cut Line= 6
      1964238.58      13564376.5      1963744.17     13562598.13
      1963817.09     13562500.91       1963865.7     13562434.94
      1963830.98     13562393.27      1963529.42     13562102.11
#Sta/Elev= 30
  2922.8  663.95    3213     659  3326.1  658.08  3349.9  658.68  3439.2  656.41
    3518  655.96  3625.9  653.68  3879.2  651.21    3960  649.19  4259.8  648.72
  4304.8  649.87  4346.3  648.93    4419  649.45  4616.2  648.28    4707  648.66
  4730.3  649.88  4740.7  649.27  4746.4  647.47  4761.5  645.28  5054.2   644.9
  5054.7   644.1  5060.7   644.1  5061.2   644.9    5086  645.39  5092.9  646.87
  5114.3   648.8  5135.4  648.49  5156.7  650.75  5234.4  652.83  5445.5  661.48
#Mann= 3 ,-1 , 0
  2922.8      .1       0  5054.2     .07       0  5061.2      .1       0
Bank Sta=5054.2,5061.2
XS Rating Curve= 0 ,0
Exp/Cntr=0.3,0.1

Type RM Length L Ch R = 1 ,23436   ,38,38,38
BEGIN DESCRIPTION:
Mapping XS 49709a14
END DESCRIPTION:
XS GIS Cut Line= 6
      1964297.17     13564428.58      1963789.31     13562695.35
      1963817.09     13562559.94      1963896.95     13562462.71
      1963907.37     13562396.74      1963563.62     13562042.58
#Sta/Elev= 30
  2823.2  664.16  3200.6  658.06  3311.3  657.51  3378.1   656.1  3383.3  656.74
  3389.6  655.52  3837.7  650.87  3910.5  649.02  4054.6  648.29  4275.9  649.54
  4304.1  648.62  4376.1  649.38    4587  648.08  4690.9  648.58  4776.3  651.07
  4876.7  651.08  4883.2  650.24  4971.5  650.91  4977.3  649.59  4993.2  650.95
  5078.4  652.33  5098.9  651.56  5131.3  647.91  5131.8  647.11  5137.8  647.11
  5138.3  647.91  5155.7  650.01  5169.9  649.94  5190.9  651.48    5463   660.9
#Mann= 3 ,-1 , 0
  2823.2      .1       0  5131.3     .07       0  5138.3      .1       0
Bank Sta=5131.3,5138.3
XS Rating Curve= 0 ,0
Exp/Cntr=0.3,0.1

Type RM Length L Ch R = 1 ,23398   ,490,490,490
BEGIN DESCRIPTION:
Mapping XS 5c3b823f
END DESCRIPTION:
XS GIS Cut Line= 6
      1964314.53     13564428.56      1963827.51     13562716.19
      1963945.56     13562459.24      1963949.03     13562365.49
      1963782.37     13562240.49      1963636.51     13562025.18
#Sta/Elev= 30
  2789.4  663.98  3198.6  657.43  3317.9  656.63  3375.3  654.96  3416.9  655.65
  3437.7   654.3  3801.6  650.99  3901.5  648.85  4490.2  648.91    4741  646.57
  4863.1  647.21  4912.7  649.01    4950  646.05  4973.2   645.4  4973.7   644.6
  4979.7   644.6  4980.2   645.4  4990.9  649.25  4997.5  648.33  5005.1  650.18
  5011.8  648.17  5019.4  649.87    5026  647.63  5033.6  648.64  5040.3  646.71
  5047.9  647.53  5054.5  646.49  5120.7  647.69  5241.5  653.46  5421.2   659.2
#Mann= 3 ,-1 , 0
  2789.4      .1       0  4973.2     .07       0  4980.2      .1       0
Bank Sta=4973.2,4980.2
XS Rating Curve= 0 ,0
Exp/Cntr=0.3,0.1

Type RM Length L Ch R = 1 ,22908   ,33,33,33
BEGIN DESCRIPTION:
Mapping XS 1c162e10
END DESCRIPTION:
XS GIS Cut Line= 6
      1964608.24     13564120.04      1964061.37     13562232.03
      1964109.11     13562193.31       1964334.8     13562158.24
      1964347.82     13562062.76      1964230.82     13561629.41
#Sta/Elev= 30
  2715.9  657.88  2825.3  657.35  3281.4  648.02  3439.5  648.06  3498.5  646.17
  3821.7  645.71  3876.8  647.35  3918.4  646.32  4012.1  647.42  4345.3  644.05
  4617.9  645.92  4657.6  644.78  4696.6  646.47  4703.1  644.55    4711  646.33
  4717.4     644  4731.8  646.42  4737.7  643.87  4758.7  645.83  4763.8  643.81
  4825.1  645.05  4830.2   643.7  4856.9  643.51  4857.4  642.71  4863.9  643.51
  4956.6  644.44  5059.9  643.56  5349.6  661.55  5432.4  664.02  5521.1  664.23
#Mann= 3 ,-1 , 0
  2715.9      .1       0  4856.9     .07       0  4863.9      .1       0
Bank Sta=4856.9,4863.9
XS Rating Curve= 0 ,0
Exp/Cntr=0.3,0.1

Type RM Length L Ch R = 1 ,22875   ,53,53,53
BEGIN DESCRIPTION:
UNT 033 in BCW 8.0
END DESCRIPTION:
XS GIS Cut Line= 6
      1964668.26     13564139.93      1964100.43     13562214.67
      1964349.99     13562188.63      1964367.36     13562169.09
      1964382.55     13562047.57      1964265.35     13561620.02
#Sta/Elev= 30
  2679.8  657.53  2820.5  657.18  3049.8   652.1  3143.7  651.48  3268.8  647.69
  3425.2  647.52  3477.3  645.88  3810.9  645.49  3863.1  647.24  3904.8  645.91
    4009  646.87  4349.6  643.74  4350.1  642.94  4356.6  643.74  4634.6  645.83
  4665.9  644.84  4684.3   647.3  4742.2  647.58  4922.9  646.15  4943.8  645.79
  4951.4   644.3  4958.1  645.52  4984.5  643.95  4989.5  645.96  5070.1  647.42
  5095.4  645.65  5255.2  656.31  5379.7  662.07  5471.2  663.71    5530  663.41
#Mann= 3 ,-1 , 0
  2679.8      .1       0  4349.6     .07       0  4356.6      .1       0
Bank Sta=4349.6,4356.6
XS Rating Curve= 0 ,0
Exp/Cntr=0.3,0.1

Type RM Length L Ch R = 1 ,22822   ,724,724,724
BEGIN DESCRIPTION:
Mapping XS 068620ce
END DESCRIPTION:
XS GIS Cut Line= 6
      1964690.71     13564072.33      1964143.83     13562253.73
      1964330.46     13562236.37      1964408.59     13562184.29
      1964430.29     13562114.84      1964317.44     13561646.07
#Sta/Elev= 30
  2765.7  657.16  2938.5  655.52  3075.8  651.85  3170.2  651.19  3284.4  647.55
  3441.7  647.13  3483.4  645.73  3838.5  645.34  3882.4  646.99  3942.9  645.67
  4019.7  646.45  4151.7  645.96  4256.2  644.03  4332.6  644.32  4381.5   643.4
    4653  645.64  4932.3  641.48  4932.8  640.68  4938.8  640.68  4939.3  641.48
  5018.3  641.75  5063.9  643.77  5090.7  646.18  5131.8  646.94  5147.7  648.48
  5189.7  648.69  5194.8  650.45  5255.2  655.67  5404.5  662.25    5501  662.44
#Mann= 3 ,-1 , 0
  2765.7      .1       0  4932.3     .07       0  4939.3      .1       0
Bank Sta=4932.3,4939.3
XS Rating Curve= 0 ,0
Exp/Cntr=0.3,0.1

Type RM Length L Ch R = 1 ,22098   ,303,303,303
BEGIN DESCRIPTION:
UNT 033 in BCW 7.0
END DESCRIPTION:
XS GIS Cut Line= 3
      1964963.83     13564057.89      1965044.52     13562073.82
      1964624.97     13561774.98
#Sta/Elev= 30
  3365.3  655.58  3418.2  655.79  3488.8  654.46  3515.2  653.07  3520.2  653.88
  3587.4  652.58  3658.4  650.61  3728.5  649.98  3788.5  647.75  4006.5  644.62
  4011.5  645.07  4028.7  644.17    4399  642.56  4589.2  640.65  4769.6   639.8
  5066.1   638.5  5066.6   637.7  5072.6   637.7  5073.1   638.5  5119.6   639.1
  5199.7  638.81  5249.7  639.76  5299.8  639.12  5392.7  639.23  5564.9  642.35
  5694.2  646.89  5787.4  652.76    5823  655.78  5843.9  656.08  5866.1  657.93
#Mann= 6 ,-1 , 0
  3365.3     .05       0  3488.8     .08       0  3587.4     .05       0
  4769.6      .1       0  5066.1     .07       0  5073.1      .1       0
Bank Sta=5066.1,5073.1
XS Rating Curve= 0 ,0
Exp/Cntr=0.3,0.1

Type RM Length L Ch R = 1 ,21795   ,1034,1034,1034
BEGIN DESCRIPTION:
UNT 033 in BCW 6.0
END DESCRIPTION:
XS GIS Cut Line= 3
      1965125.29     13564068.32      1965232.02     13561886.32
      1964846.57       13561454.
#Sta/Elev= 30
  3191.2  652.71  3288.6  652.43  3464.8   650.5  3544.9  648.45    3635  645.23
  3795.2  642.57  4315.9  639.07  4365.9  640.02    4426  639.74  4513.4  640.52
  4566.2  639.83  4696.3  640.05  4776.4  639.05  4876.5  635.95  5023.2   635.6
  5023.7   634.8  5029.7   634.8  5030.2   635.6  5176.9  636.87    5374  636.96
  5454.9  638.08  5530.4  640.86  5597.7  642.12  5644.1  643.14  5693.4   646.1
  5771.2   648.8  5778.7  649.58  5806.3  649.23  5834.7  650.25    5955  649.55
#Mann= 5 ,-1 , 0
  3191.2      .1       0  5023.2     .07       0  5030.2      .1       0
  5454.9     .05       0  5597.7      .1       0
Bank Sta=5023.2,5030.2
XS Rating Curve= 0 ,0
Exp/Cntr=0.3,0.1

Type RM Length L Ch R = 1 ,20761   ,34,34,34
BEGIN DESCRIPTION:
Mapping XS 44062390
END DESCRIPTION:
XS GIS Cut Line= 6
      1965625.29     13563708.95      1965679.98     13562146.44
      1965781.85     13561769.31       1966005.8     13561672.96
      1965599.55     13561730.25      1964932.91     13561113.08
#Sta/Elev= 30
  2788.2  647.79  3302.5  638.16  3852.8  635.68    4436  636.58  4629.3  633.22
  4629.8  632.42  4636.4  633.22  4658.6  633.44  4705.3  638.94  4738.4  636.32
    4742  633.72  4781.7  636.36  4786.8  634.06  4823.5  636.33  4827.5  634.79
  4856.9  636.01  4862.1  634.24  4889.3  636.82    4901  634.06  5072.7  633.69
    5138  633.38  5356.6   633.4  5382.2  636.56  5387.5  635.13  5413.1  636.98
  5592.3  637.28  5736.4  640.06  5833.4  642.38  6074.3  640.71    6353   643.6
#Mann= 7 ,-1 , 0
  2788.2      .1       0  4629.3     .07       0  4636.4      .1       0
  5072.7     .05       0    5138      .1       0  5592.3     .05       0
  5736.4      .1       0
Bank Sta=4629.3,4636.4
XS Rating Curve= 0 ,0
Exp/Cntr=0.3,0.1

Type RM Length L Ch R = 1 ,20727   ,60,60,60
BEGIN DESCRIPTION:
UNT 033 in BCW 5.0
END DESCRIPTION:
XS GIS Cut Line= 6
        1965675.     13563675.02      1965733.76     13561967.92
      1966048.34     13561631.12      1965657.71     13561679.73
      1965499.73     13561169.31      1964874.98     13560474.98
#Sta/Elev= 30
  2837.3  646.79    3273  638.87  3577.8  635.71  3887.9  635.12  4188.1  637.06
  4528.3  635.79    4652  632.91  4652.5  632.11  4659.1  632.91  4729.7   639.5
  4753.3  636.83  4782.3  638.48  4829.5  636.39  4851.1  637.58    4867  634.71
  4872.7  636.69  4903.6  636.87  4926.2  636.31  4931.9  634.14  5003.6  635.95
  5103.2  634.57  5121.9  636.28  5217.3  636.05    5325   638.7  5521.6  636.29
  5648.9  637.06  5783.3  639.44  6012.7  637.25  6260.1  639.71    6919  653.95
#Mann= 7 ,-1 , 0
  2837.3      .1       0    4652     .07       0  4659.1      .1       0
  5121.9     .05       0  5217.3      .1       0  5521.6     .05       0
  5648.9      .1       0
Bank Sta=4652,4659.1
XS Rating Curve= 0 ,0
Exp/Cntr=0.3,0.1

Type RM Length L Ch R = 1 ,20667   ,598,598,598
BEGIN DESCRIPTION:
Mapping XS f436bab6
END DESCRIPTION:
XS GIS Cut Line= 6
      1965716.74     13563678.71       1965815.7      13561876.6
      1966044.87     13561756.81      1966096.95     13561600.56
      1965685.49     13561605.77      1965206.95     13560248.18
#Sta/Elev= 30
  2811.7  646.52  2985.7  644.76  3286.1  638.25  3556.5  635.55  3776.9  635.49
    3857  634.22  4027.2  636.19  4387.8  636.17  4734.6  632.91  4752.4  633.63
  4808.2  631.99  4886.9  632.45  4950.7  631.33  4952.6  630.56  4953.1  629.76
  4959.2  629.76  4959.7  630.56  5093.7  632.68  5118.8  633.72  5314.1  633.98
  5504.8   636.7    5609   636.2    5747  639.18  6008.5  636.99  6146.3  638.81
  6178.2  638.16  6200.6  638.44    6210  639.87  6326.6  640.91  6927.6  643.68
#Mann= 5 ,-1 , 0
  2811.7      .1       0  4952.6     .07       0  4959.7      .1       0
  5093.7     .05       0    5609      .1       0
Bank Sta=4952.6,4959.7
XS Rating Curve= 0 ,0
Exp/Cntr=0.3,0.1

Type RM Length L Ch R = 1 ,20069   ,963,963,963
BEGIN DESCRIPTION:
UNT 033 in BCW 4.0
END DESCRIPTION:
XS GIS Cut Line= 3
      1966858.34     13562879.92      1966841.87     13561641.82
       1965806.7     13560565.42
#Sta/Elev= 30
  3366.9  632.35  3391.8  632.91  3401.8  631.86  3431.8  631.48  3441.8  632.69
  3481.8   632.9  3534.4  630.83  3571.8     631  3641.8   629.3  4088.3  627.77
  4088.8  626.97  4094.9  626.97  4095.4  627.77  4311.9  628.13  4431.9   629.4
  4511.9  628.79  4571.9  629.66  4591.9   630.8  4609.2  629.93  4650.2  629.38
  4848.3  630.28  5003.7  628.17    5032  628.44  5088.6  630.37  5216.7  629.94
  5364.3  628.96  5438.8  629.79  5555.5  629.75  5696.7  632.48  6098.5  636.45
#Mann= 7 ,-1 , 0
  3366.9     .05       0  3534.4      .1       0  4088.3     .03       0
  4095.4      .1       0  4609.2     .05       0  5216.7      .1       0
  5438.8     .05       0
Bank Sta=4088.3,4095.4
XS Rating Curve= 0 ,0
Exp/Cntr=0.3,0.1

Type RM Length L Ch R = 1 ,19106   ,124,124,124
BEGIN DESCRIPTION:
Mapping XS 3fabe7cb
END DESCRIPTION:
XS GIS Cut Line= 3
      1966873.04     13562940.06      1966943.45     13561530.45
      1966892.95     13560183.66
#Sta/Elev= 30
  2612.2  632.44  2651.6  632.57  2717.4  632.44  2737.4   631.4  2767.5  631.34
  2787.5  632.85  2874.2  630.84  2937.7  629.29  3127.9  628.21  3338.2  628.36
  3553.5  627.29  3718.6  628.57  3858.8  628.66  3908.9  629.85    3921  629.35
  3954.1  628.29  4099.1  628.98  4429.3  627.87  4539.4  628.43  4608.5  627.39
  4769.5  624.94  4915.5  625.48  4975.8  624.53  4976.4  623.73  4982.9  623.73
  4983.6  624.53  5039.7  626.14  5076.5  628.41  5189.8  633.17  5371.3   636.2
#Mann= 8 ,-1 , 0
  2612.2      .1       0  2651.6     .05       0  2874.2      .1       0
    3921     .05       0  4608.5      .1       0  4975.8     .07       0
  4983.6      .1       0  5076.5     .05       0
Bank Sta=4975.8,4983.6
XS Rating Curve= 0 ,0
Exp/Cntr=0.3,0.1

Type RM Length L Ch R = 1 ,18982   ,370,370,370
BEGIN DESCRIPTION:
Mapping XS 66128a51
END DESCRIPTION:
XS GIS Cut Line= 3
      1966886.92     13562936.63      1967105.68     13561555.24
      1966997.11     13560235.71
#Sta/Elev= 30
  2545.4  632.61  2606.5  632.27  2698.9  632.19  2729.3  630.75  2749.5  631.82
  2865.4   629.2  3449.9   627.2    3519     628  3529.1   626.8  3630.4  626.57
  3648.8  626.66  3653.8  627.92    3681  627.22  3701.3  628.13  3716.2  627.09
  3762.8  627.23  4011.4  626.82  4044.6  628.33  4084.7  626.76  4215.2  627.56
  4375.3  626.66  4566.3  627.05  4754.6  625.83  4827.2  626.36  4907.5  624.39
  4993.9  624.14  4994.5  623.34  5001.7  624.14    5112  629.48    5268  633.47
#Mann= 9 ,-1 , 0
  2545.4      .1       0  2606.5     .05       0  2865.4      .1       0
  3449.9     .05       0  3762.8      .1       0  4375.3     .05       0
  4754.6      .1       0  4993.9     .07       0  5001.7      .1       0
Bank Sta=4993.9,5001.7
XS Rating Curve= 0 ,0
Exp/Cntr=0.3,0.1

Type RM Length L Ch R = 1 ,18612   ,501,501,501
BEGIN DESCRIPTION:
Mapping XS 8db6c047
END DESCRIPTION:
XS GIS Cut Line= 4
      1966884.85     13562950.81      1967399.89     13561214.92
      1967386.01     13560503.11      1967153.73      13560149.5
#Sta/Elev= 30
  2478.8  631.82  2493.5  632.61  2575.3  631.77  2662.2  631.79  2693.5  630.16
  2735.2  629.36  2741.7  630.05  2746.9  629.14  2756.1  629.86    2996  627.76
  3110.7  628.13  3298.5  626.15  3309.8  625.38  3402.8  626.37  3423.6  625.01
  3442.7  626.12  3507.1  625.21  3997.3  625.45  4187.3  624.16  4629.5   623.8
  4959.5  622.87  4985.6  621.69  4986.3  620.89  4992.8  620.89  4993.4  621.69
  5035.8  623.38  5081.1  622.76  5138.3   623.7    5304  629.32  5424.5  631.09
#Mann= 5 ,-1 , 0
  2478.8      .1       0  2575.3     .05       0  3298.5      .1       0
  4985.6     .07       0  4993.4      .1       0
Bank Sta=4985.6,4993.4
XS Rating Curve= 0 ,0
Exp/Cntr=0.3,0.1

Type RM Length L Ch R = 1 ,18111   ,464,464,464
BEGIN DESCRIPTION:
Mapping XS 89d9033a
END DESCRIPTION:
XS GIS Cut Line= 4
      1966900.46     13562956.06      1967826.98     13560912.83
      1967792.26     13560187.14      1967114.57     13559659.62
#Sta/Elev= 30
  2136.3  631.35  2156.7  632.32    2260  630.41  2306.2  630.02  2327.3  630.84
  2450.2  627.91  2478.8  629.23  2496.4  628.18  2583.3   627.7  2720.6  625.83
  2910.8  625.89  3147.2  624.15  3169.6  624.83  3839.4   622.3  4015.1  622.54
  4397.6  620.43  4803.3  620.45  4948.8  620.37  4997.4  619.34  5004.4  619.08
  5005.1  618.28  5011.6  618.28  5012.2  619.08  5068.4  620.82  5098.4  619.36
  5177.8  620.61  5362.4  619.83  5455.6  621.31  5526.1  621.38  5965.1  630.14
#Mann= 7 ,-1 , 0
  2136.3      .1       0  2327.3     .05       0  2583.3      .1       0
  4803.3     .12       0  4997.4      .1       0  5004.4     .07       0
  5012.2      .1       0
Bank Sta=5004.4,5012.2
XS Rating Curve= 0 ,0
Exp/Cntr=0.3,0.1

Type RM Length L Ch R = 1 ,17647   ,385,385,385
BEGIN DESCRIPTION:
Mapping XS c7c93904
END DESCRIPTION:
XS GIS Cut Line= 4
      1966900.48     13563013.32      1968147.72     13560964.05
      1968145.55     13560488.79      1967224.71     13559618.76
#Sta/Elev= 30
  2181.5  631.14  2262.4  630.23    2272  630.96  2357.3  628.93  2446.4  628.52
  2547.2  626.48    2584   627.2  2605.3  626.25  2721.5  625.27  3092.6  625.13
  3275.5  623.24  3361.9  623.78  3755.9   621.1  4089.2  620.62  4315.8  618.57
  4959.5  618.22  4995.6  616.63  4996.3  615.83  5002.8  615.83  5003.4  616.63
  5049.5   618.9  5157.8  619.84  5214.4  618.94  5455.1  620.08  5476.2  620.03
  5483.1  619.18    5547  620.26  5829.8  619.59  6091.5  622.69  6322.6   627.5
#Mann= 3 ,-1 , 0
  2181.5      .1       0  4995.6     .07       0  5003.4      .1       0
Bank Sta=4995.6,5003.4
XS Rating Curve= 0 ,0
Exp/Cntr=0.3,0.1

Type RM Length L Ch R = 1 ,17262   ,1086,1086,1086
BEGIN DESCRIPTION:
Mapping XS a3c11d74
END DESCRIPTION:
XS GIS Cut Line= 4
      1966879.65     13563091.44      1968697.34     13560909.18
      1968395.26     13560268.55      1967209.01     13559550.56
#Sta/Elev= 30
  1690.4  630.01    1827   629.8    1883   628.4  1890.8  629.22  1961.1  627.46
  2018.4  627.99  2039.2  626.27  2238.3  624.25  2735.6  623.94  2976.4  622.04
  3118.3  622.38  3232.9  620.29  3715.9  619.31  3872.1  618.03  4361.5  617.73
  4723.1  615.64  4888.9  616.84  4977.4  615.94  4993.6  615.46  4995.6  613.84
  4996.2  613.04  5002.8  613.04  5003.4  613.84  5010.5  616.34  5084.7   617.1
    5446  616.61  5742.8  618.69  6202.5  619.26  6361.6  621.72  6625.4  627.78
#Mann= 3 ,-1 , 0
  1690.4      .1       0  4995.6     .07       0  5003.4      .1       0
Bank Sta=4995.6,5003.4
XS Rating Curve= 0 ,0
Exp/Cntr=0.3,0.1

Type RM Length L Ch R = 1 ,16176   ,641,641,641
BEGIN DESCRIPTION:
Mapping XS 8bc35be2
END DESCRIPTION:
XS GIS Cut Line= 4
       1970854.6     13560960.52      1969880.36      13560208.2
      1968360.41     13560043.83      1967668.59     13559576.12
#Sta/Elev= 30
    2814  629.57  2838.8  628.83  2860.8  626.28    2917  623.61  3074.6   618.6
  3206.8  615.49  3352.6  613.17  3558.9  611.54  3686.8  612.61  3736.6  610.46
  3773.7  609.94  3795.3  607.36  3795.9  606.56  3805.9  606.56  3806.6  607.36
  3887.4  608.97  3964.9  611.67  4490.5  612.95  4563.3  614.36  4587.3  613.52
  4830.2  614.03  4954.4  613.28  4993.7  611.47  5005.8   610.9  5015.9  612.07
  5367.9   615.3  5408.2  614.92  5577.4  616.36  5742.2  616.05  6408.8  617.66
#Mann= 6 ,-1 , 0
    2814     .05       0  3206.8      .1       0  3795.3     .07       0
  3806.6      .1       0  4830.2     .12       0  4993.7      .1       0
Bank Sta=3795.3,3806.6
XS Rating Curve= 0 ,0
Exp/Cntr=0.3,0.1

Type RM Length L Ch R = 1 ,15535   ,66,66,66
BEGIN DESCRIPTION:
Mapping XS 7a5b3d28
END DESCRIPTION:
XS GIS Cut Line= 6
      1970932.78     13560252.22      1968965.87     13559683.67
      1968899.89     13559475.33      1968844.34     13559475.33
      1968795.73     13559701.03      1968119.31     13559756.53
#Sta/Elev= 30
  2721.3  615.02  2815.5  614.55  2854.3  617.28  2923.1  614.19  3135.4  615.64
    3195  611.99  3312.3  609.27  3364.4  610.63  3451.2  607.46  3749.5  611.87
  3951.1  611.17  4360.9  611.67  4613.5  612.32  4711.1  609.63  4744.8  611.54
  4801.8  610.13  4859.4   603.2  4899.6  605.04  4907.9  602.58  4908.6  601.78
  4919.2  602.58  4965.9  605.72  4983.7  602.73  5053.2  607.42  5085.7  605.61
  5125.3  608.08  5135.8  610.87  5241.5   612.7  5279.6  611.07  5969.1  616.29
#Mann= 7 ,-1 , 0
  2721.3      .1       0  2815.5     .05       0  2923.1      .1       0
  3951.1     .05       0  4360.9      .1       0  4907.9     .07       0
  4919.2      .1       0
Bank Sta=4907.9,4919.2
XS Rating Curve= 0 ,0
Exp/Cntr=0.3,0.1

Type RM Length L Ch R = 1 ,15469   ,39,39,39
BEGIN DESCRIPTION:
Mapping XS 7e75d2fe
END DESCRIPTION:
XS GIS Cut Line= 6
      1970833.75     13560106.37      1969000.59     13559638.53
      1968903.37     13559409.36      1968792.26     13559437.14
      1968792.26     13559621.17      1968094.37     13559707.97
#Sta/Elev= 30
  2818.7  613.96  2843.4   617.4  2889.8  615.22  2913.1  615.72  3127.7  617.23
  3241.5  613.24  3270.4  610.72  3303.6  610.82  3334.6  608.46  3385.4   607.5
  3386.1   606.7  3396.7   607.5  3541.5  610.25  3675.3  610.27  3996.7  611.85
  4399.2  611.15  4561.7  611.99  4657.6  611.04  4691.6  609.48    4719  611.49
  4836.5  614.82    4907  615.71  4953.4  614.08  4958.5  615.72  5039.4  616.78
  5085.8  615.94  5119.9   617.2    5294   616.1  5337.7  611.47  6003.4  616.02
#Mann= 6 ,-1 , 0
  2818.7     .08       0  2913.1      .1       0  3385.4     .07       0
  3396.7      .1       0  3675.3     .05       0  4399.2      .1       0
Bank Sta=3385.4,3396.7
XS Rating Curve= 0 ,0
Exp/Cntr=0.3,0.1

Type RM Length L Ch R = 1 ,15430   ,90,90,90
BEGIN DESCRIPTION:
Mapping XS c495f884
END DESCRIPTION:
XS GIS Cut Line= 6
      1970953.56     13560033.45      1969045.73     13559596.86
      1968997.12     13559364.22      1968705.45     13559409.36
      1968733.23     13559582.97      1968119.29     13559673.15
#Sta/Elev= 30
  2706.1  614.27  2819.4  615.57    2838  615.28  2854.7  617.67  2868.8  617.94
  2897.7  616.49  2919.5  617.21  2988.6  617.99  3012.4  619.84  3036.7  618.54
  3127.7  618.95  3238.1  614.05  3309.9  609.46  3396.6  606.63  3397.2  605.83
  3407.2  605.83  3407.9  606.63  3494.5  609.85  3566.4  609.74  4120.3  611.63
  4253.7  610.56  4425.4  611.01  4551.2  611.83  4661.1  610.07  4902.8  608.76
    4994  610.14  5110.4  609.93  5203.9  611.63    5374  611.65  6002.6  616.13
#Mann= 7 ,-1 , 0
  2706.1      .1       0  2819.4     .08       0  2919.5      .1       0
  3396.6     .07       0  3407.9      .1       0  3566.4     .05       0
  4425.4      .1       0
Bank Sta=3396.6,3407.9
XS Rating Curve= 0 ,0
Exp/Cntr=0.3,0.1

Type RM Length L Ch R = 1 ,15340   ,603,603,603
BEGIN DESCRIPTION:
Mapping XS c89973d4
END DESCRIPTION:
XS GIS Cut Line= 3
      1970885.92     13559903.27      1969158.97     13559262.89
      1968000.58     13559386.21
#Sta/Elev= 30
  2932.6  615.99  2974.2  617.34  2994.9  616.25  3008.2  616.45  3026.3  618.47
  3050.9  618.49  3072.2   617.1  3081.6  617.76  3104.2  619.32  3147.8  619.53
  3283.7  618.07  3392.2   614.3  3485.7  608.57  3552.2  607.21  3576.8  605.67
  3578.5   604.3  3579.2   603.5  3589.2   603.5  3589.8   604.3  3601.9  606.07
  3648.2  608.47  3712.2  609.63  3736.8  608.99  4192.1  610.48  4404.5  608.69
  4722.6  610.15  4814.4  609.27  5032.7  608.32  5160.6  610.81  5939.4  614.81
#Mann= 8 ,-1 , 0
  2932.6      .1       0  2974.2     .08       0  2994.9     .05       0
  3081.6      .1       0  3578.5     .07       0  3589.8      .1       0
  3736.8     .05       0  4814.4      .1       0
Bank Sta=3578.5,3589.8
XS Rating Curve= 0 ,0
Exp/Cntr=0.3,0.1

Type RM Length L Ch R = 1 ,14737   ,289,289,289
BEGIN DESCRIPTION:
Mapping XS 857befe7
END DESCRIPTION:
XS GIS Cut Line= 3
      1971510.84     13558726.17      1968153.24     13558779.99
      1967620.24     13559002.22
#Sta/Elev= 30
  2637.8  614.53  2673.6  614.51  2693.6  611.85  2723.6  610.71  2783.7  615.06
  2903.7  611.39  3363.9  608.19  3413.7  607.84  3433.7  609.68  3462.3  609.27
  3483.7  607.93  3628.1  608.18  3783.8  604.67  3793.8  603.86  3803.8  600.83
  3818.1  599.39  3818.8  598.59  3828.8  598.59  3829.5  599.39  3843.8  600.93
  3853.8  604.29  3863.3  604.72  4121.8  606.51  4403.9  605.16  4743.8  608.54
  4913.9  605.54  4993.9   605.2    5154  607.74  6058.9  609.82  6573.3  613.17
#Mann= 7 ,-1 , 0
  2637.8      .1       0  3363.9     .08       0  3462.3      .1       0
  3628.1     .16       0  3818.1     .07       0  3829.5     .16       0
  3863.3      .1       0
Bank Sta=3818.1,3829.5
XS Rating Curve= 0 ,0
Exp/Cntr=0.3,0.1

Type RM Length L Ch R = 1 ,14448   ,631,631,631
BEGIN DESCRIPTION:
Mapping XS 8edb3ff5
END DESCRIPTION:
XS GIS Cut Line= 4
      1971375.49     13558429.29      1970479.63     13558424.09
      1968875.59     13558545.93      1967302.58     13558757.41
#Sta/Elev= 30
    2885  612.53    2904  611.51  3175.5  607.24  3465.9  606.52  3545.5  606.09
  3564.2  607.73  3595.5  607.88  3615.5   606.1  3635.5  607.43  3662.5  607.04
  3927.2  604.99  4016.2   603.8  4030.5  599.78  4031.2  598.98  4041.2  598.98
  4041.9  599.78  4046.3  601.91  4056.3  603.97  4096.4   604.9  4120.1  604.35
    4297  604.96  4377.2  602.68  4557.7  605.71  4848.6  607.25  4968.9  604.76
  4978.9  603.78    4999  604.89  5129.4  606.47  6278.1  609.34  6976.7  614.03
#Mann= 9 ,-1 , 0
    2885      .1       0    2904     .05       0  3465.9      .1       0
  3564.2     .08       0  3662.5      .1       0  3927.2     .16       0
  4030.5     .07       0  4041.9     .16       0  4120.1      .1       0
Bank Sta=4030.5,4041.9
XS Rating Curve= 0 ,0
Exp/Cntr=0.3,0.1

Type RM Length L Ch R = 1 ,13817   ,754,754,754
BEGIN DESCRIPTION:
Mapping XS cf3ba813
END DESCRIPTION:
XS GIS Cut Line= 4
      1971604.68     13558184.51      1970339.15     13557899.89
      1968599.42     13558038.67      1967290.42     13557896.43
#Sta/Elev= 30
  2348.7  607.41  2942.9  601.75  3165.4  603.99  3265.5  605.15  3301.6  604.22
  3332.3  605.73  3365.6  604.47  3383.6  605.03  3424.6  603.28  3558.6  601.97
  3850.6  602.43  3891.6   599.9  3892.2   599.1  3902.3   599.1    3903   599.9
  3930.9  601.92  4061.3  601.35  4091.4  603.01  4221.8  604.19  4783.8  604.22
  5004.3  602.49  5158.1  604.83  5223.3  604.67  5275.1  605.02  5295.2  606.31
  5335.3  605.34  5471.2  605.38  5868.3  607.92  6381.3  613.69  6707.8  615.71
#Mann= 7 ,-1 , 0
  2348.7     .05       0  3165.4      .1       0  3265.5     .08       0
  3365.6     .05       0  3891.6    .035       0    3903     .05       0
  5223.3      .1       0
Bank Sta=3891.6,3903
XS Rating Curve= 0 ,0
Exp/Cntr=0.3,0.1

Type RM Length L Ch R = 1 ,13063   ,515,515,515
BEGIN DESCRIPTION:
Mapping XS bb4ffef4
END DESCRIPTION:
XS GIS Cut Line= 3
      1971635.89     13558028.26       1969583.8     13557460.54
      1967911.02     13556937.22
#Sta/Elev= 30
  2574.3  605.35  3062.9  599.89    3383  601.81  3527.9   603.2  3583.6  602.19
  3612.7  604.61  3657.4  601.89  4058.9  601.56  4125.9  598.06  4126.5  597.26
  4137.3  598.06  4245.7  602.27  4619.2  602.94  4995.6  600.89  5329.6  602.97
  5738.9  605.14    5750  603.71  5773.1  604.83  5846.8  606.04  5981.9  609.03
  6041.6  608.82  6079.3  610.57  6111.7   609.7    6117  611.09  6209.1   612.4
  6279.3  617.89  6284.5  619.61  6311.8  620.86    6317  622.99  6456.2  621.22
#Mann= 8 ,-1 , 0
  2574.3     .05       0    3383      .1       0  3527.9     .05       0
  4125.9    .035       0  4137.3     .05       0  5329.6      .1       0
  5773.1     .16       0  5846.8      .1       0
Bank Sta=4125.9,4137.3
XS Rating Curve= 0 ,0
Exp/Cntr=0.3,0.1
