HEC-RAS study CHACON CREEK.prj: CHACON CREEK Base Level Engineering

--- CHACON CREEK.g01 (geometry) --- (continued)

Type RM Length L Ch R = 1 ,150559  ,177,177,177
BEGIN DESCRIPTION:
CHACON CREEK 203.0
END DESCRIPTION:
XS GIS Cut Line= 3
      1987695.79     13674474.54       1987306.9     13674460.65
      1986133.29     13674450.24
#Sta/Elev= 30
  4296.3  914.72  4387.2  913.09  4417.2  912.09  4427.9  911.22 4456.22910.3349
  4487.2  909.46  4517.2  909.33  4577.3  908.45  4637.3  908.27  4657.3  908.46
    4680  908.22  4680.6  907.42  4687.1  907.42  4687.7  908.22  4755.6  908.27
  4760.6  909.64  4797.3  909.49  4857.3  910.04  4927.4  910.14  4977.4  910.52
  5037.4  909.93  5072.5  909.95 5215.11910.3348  5269.3  910.61  5367.7  911.32
  5473.8  912.23  5527.4  912.79  5557.6   913.4  5677.4  916.16  5859.1  922.46
#Mann= 8 ,-1 , 0
  4296.3     .05       0    4680     .04       0  4687.7     .05       0
  5072.5     .08       0  5269.3     .05       0  5367.7     .08       0
  5473.8      .1       0  5557.6     .08       0
Bank Sta=4456.22,5215.11
XS Rating Curve= 0 ,0
Exp/Cntr=0.3,0.1

Type RM Length L Ch R = 1 ,150382  ,273,273,273
BEGIN DESCRIPTION:
CHACON CREEK 202.0
END DESCRIPTION:
XS GIS Cut Line= 3
      1987737.42     13674283.57      1987327.73     13674276.62
      1986148.56      13674290.5
#Sta/Elev= 30
  4253.1  913.03  4462.1   911.4  4467.1  909.37  4572.9  908.62 4660.21908.0593
  4815.6  906.86  4915.6  906.55  4940.6  906.12  4941.5  905.32    4949  905.32
  4949.9  906.12  4950.2  907.75  4985.6  907.29  4995.6  907.75  5005.6  906.71
  5015.6  906.65  5035.6  907.55  5075.6  907.19 5133.53908.0593  5265.6  908.77
  5285.6  909.14  5315.6  908.59  5360.6  908.57  5515.6  909.47  5585.6  910.54
    5656  912.41  5685.7  913.04  5795.3  917.87  5800.3  917.53  5842.1  919.78
#Mann= 6 ,-1 , 0
  4253.1     .05       0  4572.9      .1       0  4940.6     .07       0
  4949.9      .1       0  5360.6     .08       0    5656     .05       0
Bank Sta=4660.21,5133.53
XS Rating Curve= 0 ,0
Exp/Cntr=0.3,0.1

Type RM Length L Ch R = 1 ,150109  ,306,306,306
BEGIN DESCRIPTION:
CHACON CREEK 201.0
END DESCRIPTION:
XS GIS Cut Line= 3
      1987874.27     13674277.63      1987202.73      13674116.9
      1986390.23     13673734.96
#Sta/Elev= 30
    4186   913.1  4214.9  912.95    4220  911.28  4351.3  907.07  4468.6  905.72
  4551.5  905.46 4775.78 904.204  4929.2  902.21  4965.6  899.76  4982.9  900.12
  4990.9  898.09  4991.8  897.29  5000.2  898.09  5017.6  902.33  5072.9  902.92
  5117.1  905.18  5130.7  905.14    5148  903.01  5153.5  904.96  5170.8  904.85
  5176.3   906.2  5199.1  904.18  5243.3  904.27  5250.3  902.32  5273.1  900.97
  5300.4  902.18 5401.09904.2042  5414.4  904.43  5496.3  906.08  5774.3  913.88
#Mann= 9 ,-1 , 0
    4186     .05       0  4468.6     .16       0  4551.5      .1       0
  4990.9     .07       0  5000.2      .1       0  5243.3     .16       0
  5300.4      .1       0  5414.4     .16       0  5496.3      .1       0
Bank Sta=4775.78,5401.09
XS Rating Curve= 0 ,0
Exp/Cntr=0.3,0.1

Type RM Length L Ch R = 1 ,149803  ,229,229,229
BEGIN DESCRIPTION:
Mapping XS 6bc931c8
END DESCRIPTION:
XS GIS Cut Line= 3
      1987900.26     13674245.05       1986801.6     13673518.46
      1986529.12     13673492.51
#Sta/Elev= 30
  4259.8  910.29    4305  908.67    4415  905.07  4538.3  903.86  4665.2  903.38
    4740  902.93 4796.16901.6125  4863.4   900.2  4879.8  897.13  4880.7  896.33
  4888.2  896.33  4889.1  897.13  4920.5  900.13  4956.7  900.48  4973.2  899.09
  4992.8  897.52  4998.8   897.9  5013.8  901.14  5049.9  902.07  5137.2  900.63
  5158.3   898.1  5188.4  900.18  5209.4  899.78  5251.5  901.42 5353.16901.6124
  5467.8  902.75  5583.6  903.79  5623.8  905.54  5764.4  908.97  5850.7   912.3
#Mann= 8 ,-1 , 0
  4259.8     .05       0    4305      .1       0  4538.3     .16       0
  4665.2      .1       0  4879.8     .07       0  4889.1      .1       0
  4973.2     .16       0  5467.8      .1       0
Bank Sta=4796.16,5353.16
XS Rating Curve= 0 ,0
Exp/Cntr=0.3,0.1

Type RM Length L Ch R = 1 ,149574  ,355,355,355
BEGIN DESCRIPTION:
Mapping XS 79a27b46
END DESCRIPTION:
XS GIS Cut Line= 3
      1987904.66     13674236.42      1987369.31     13673583.79
      1987181.81     13672430.14
#Sta/Elev= 30
  4299.6  909.89  4319.5  908.81  4463.9   904.5  4586.2  903.08  4733.7  902.39
  4818.8  901.17 4849.48899.8056  4883.5  898.96    4911  897.13  4920.7  895.12
  4921.5  894.32  4929.1  894.32    4930  895.12  4933.2  896.91  4939.7  898.55
  4947.5   898.7  4974.8  898.44  4997.1  896.07  5017.9   897.8  5081.7  899.42
  5213.6  897.63  5253.9  897.03  5261.5  895.59  5343.4   898.5  5377.4  899.67
 5390.11899.8054  5512.8  903.27  5764.2  907.57    6072  917.37  6312.5  921.95
#Mann= 8 ,-1 , 0
  4299.6     .05       0  4319.5      .1       0  4586.2     .16       0
  4920.7     .07       0    4930     .16       0  5213.6      .1       0
  5343.4     .16       0  5377.4      .1       0
Bank Sta=4849.48,5390.11
XS Rating Curve= 0 ,0
Exp/Cntr=0.3,0.1

Type RM Length L Ch R = 1 ,149219  ,356,356,356
BEGIN DESCRIPTION:
CHACON CREEK 200.0
END DESCRIPTION:
XS GIS Cut Line= 3
       1987981.3     13674091.62        1987725.       13673525.
      1987525.01     13672925.04
#Sta/Elev= 30
  4333.2  907.16  4456.7  902.98  4705.4  900.51  4842.9  899.06  4856.3   899.6
    4888898.4877  4940.8  897.04  4965.6  894.77  4976.2  892.99  4986.7  893.67
  5007.8   893.2  5018.3  894.42  5028.9  894.33  5039.4  896.32  5081.6  897.47
  5155.4  895.05  5165.9  893.65  5176.4  893.82    5187  892.65  5192.9     891
  5193.7   890.2  5201.3   890.2  5202.2     891 5236.51898.4877  5260.8  900.84
    5324  903.28  5418.9  904.79  5479.4  906.72  5485.2  906.98  5587.5  910.54
#Mann= 7 ,-1 , 0
  4333.2      .1       0  4705.4     .16       0  5039.4      .1       0
  5192.9     .07       0  5202.2      .1       0  5479.4     .16       0
  5485.2      .1       0
Bank Sta=4888,5236.51
XS Rating Curve= 0 ,0
Exp/Cntr=0.3,0.1

Type RM Length L Ch R = 1 ,148863  ,334,334,334
BEGIN DESCRIPTION:
CHACON CREEK 199.0
END DESCRIPTION:
XS GIS Cut Line= 3
        1988275.     13674224.99        1987875.       13673225.
      1987725.01     13672925.03
#Sta/Elev= 30
  3900.1  912.15  4232.6  902.67  4342.7  901.15  4470.9  900.69  4567.8  899.46
 4663.31897.1847  4693.1  896.02  4771.1  894.66  4807.6  895.11  4858.1  895.34
  4955.6  895.63  4967.7   894.8  4974.4  893.09  4979.9  893.09  4985.5  891.91
  4991.1  891.86  4999.5  889.18  5008.5  888.96  5009.5  888.16  5017.5  888.16
  5018.4  888.96  5021.8  890.73  5030.2  892.41  5052.6  896.05  5058.2  895.95
 5067.77897.1849    5112  898.75    5142  899.45  5237.1  905.36  5312.5  907.37
#Mann= 7 ,-1 , 0
  3900.1      .1       0  4342.7     .16       0  4807.6      .1       0
  4858.1     .16       0  5008.5     .07       0  5018.4     .16       0
    5112      .1       0
Bank Sta=4663.31,5067.77
XS Rating Curve= 0 ,0
Exp/Cntr=0.3,0.1

Type RM Length L Ch R = 1 ,148529  ,516,516,516
BEGIN DESCRIPTION:
CHACON CREEK 198.0
END DESCRIPTION:
XS GIS Cut Line= 3
      1988429.19     13674151.45        1988175.       13673225.
        1987825.       13672825.
#Sta/Elev= 30
  4049.2  910.26  4082.9  909.09  4211.4  907.54    4350  902.22  4588.5  900.06
  4844.5   897.5  4864.7  896.84 4867.66896.0236  4878.9  893.58  4885.5  890.79
  4895.8  890.12  4926.9  890.45  4968.4  892.11  4978.8  891.22  4982.5  887.75
  4983.5  886.95  4991.5  886.95  4992.4  887.75  4992.7     889  4999.5  888.22
  5007.3  891.42  5013.2  891.42    5017  893.47  5023.7  892.42  5031.2  893.54
  5109.1  893.76 5193.67896.0236    5315  898.41  5386.3  901.26  5541.4  907.68
#Mann= 5 ,-1 , 0
  4049.2      .1       0  4588.5     .16       0  4982.5     .07       0
  4992.4     .16       0  5386.3      .1       0
Bank Sta=4867.66,5193.67
XS Rating Curve= 0 ,0
Exp/Cntr=0.3,0.1

Type RM Length L Ch R = 1 ,148013  ,281,281,281
BEGIN DESCRIPTION:
CHACON CREEK 197.0
END DESCRIPTION:
XS GIS Cut Line= 3
      1989174.01     13673734.84       1988489.1     13673052.54
      1987975.01     13672625.01
#Sta/Elev= 30
  3957.4  915.16  4041.4  912.92  4084.6  911.01  4105.1  909.77  4274.8  904.21
    4296  903.02  4501.1  900.26  4663.7  896.52  4684.9  895.21    4692  895.78
  4721.3  894.12 4755.39893.3883  4840.5  891.62  4932.1  890.96  4939.9  889.81
  4960.7  888.56  4976.4  884.72  4977.4  883.92  4985.7  883.92  4986.6  884.72
  4995.9  885.04  5003.7  888.43    5018  890.98  5038.8  891.33 5073.39893.3884
  5252.4  896.36  5266.7  896.75    5294  898.92  5338.6  900.33  5592.8  910.33
#Mann= 6 ,-1 , 0
  3957.4     .16       0  4084.6      .1       0  4721.3     .16       0
  4976.4     .07       0  4986.6     .16       0  5338.6      .1       0
Bank Sta=4755.39,5073.39
XS Rating Curve= 0 ,0
Exp/Cntr=0.3,0.1

Type RM Length L Ch R = 1 ,147732  ,382,382,382
BEGIN DESCRIPTION:
CHACON CREEK 196.0
END DESCRIPTION:
XS GIS Cut Line= 3
        1989525.       13673775.        1988525.       13672775.
      1988174.99     13672424.99
#Sta/Elev= 30
  3554.2  927.02  3794.6  916.45  3905.2  912.79  3950.2  911.38  4020.9  907.07
  4063.3   906.4    4134   902.8  4416.9  896.38  4459.3  894.87  4501.7  892.22
 4534.83891.4494  4600.7  890.37  4667.5  890.37  4742.1  891.09  4855.3  887.77
  4883.6  888.88  4911.8  887.43    4926  888.07    4935  886.26    4936  885.46
  4944.3  885.46  4945.2  886.26  4964.9  888.62  5010.8  886.44 5022.78891.4513
  5039.1  894.71  5072.4  894.77  5128.9  895.63  5194.7   897.1  5463.4  913.45
#Mann= 7 ,-1 , 0
  3554.2     .16       0  3905.2      .1       0  4667.5     .16       0
    4935     .07       0  4945.2     .16       0  5072.4      .1       0
  5128.9     .16       0
Bank Sta=4534.83,5022.78
XS Rating Curve= 0 ,0
Exp/Cntr=0.3,0.1

Type RM Length L Ch R = 1 ,147350  ,371,371,371
BEGIN DESCRIPTION:
CHACON CREEK 195.0
END DESCRIPTION:
XS GIS Cut Line= 3
      1989324.99     13673224.99        1988875.       13672725.
      1988424.97     13672224.96
#Sta/Elev= 30
  4299.8  902.95  4377.9  899.52  4512.4  896.52 4617.31889.8162  4682.1  888.02
    4774  889.77  4835.5  889.24  4851.8  887.39  4859.2  885.41  4922.8  885.24
  4930.2   883.5    4937  884.42  4939.3  882.55  4940.3  881.75  4948.6  881.75
  4949.5  882.55  4951.2  883.66  4958.6  882.69  4965.4  883.52  5014.7  883.58
  5022.2  887.72  5028.9  888.12 5033.66889.8146  5036.4  890.79  5071.5  892.23
  5176.5  893.28  5362.3  895.09  5444.2  901.15  5633.7  911.86  5645.2   912.6
#Mann= 7 ,-1 , 0
  4299.8      .1       0  4835.5     .16       0  4939.3     .07       0
  4949.5     .16       0  5176.5      .1       0  5444.2     .16       0
  5633.7      .1       0
Bank Sta=4617.31,5033.66
XS Rating Curve= 0 ,0
Exp/Cntr=0.3,0.1

Type RM Length L Ch R = 1 ,146979  ,335,335,335
BEGIN DESCRIPTION:
CHACON CREEK 194.0
END DESCRIPTION:
XS GIS Cut Line= 3
      1989625.02     13673125.02        1989125.       13672625.
      1988625.02     13672125.02
#Sta/Elev= 30
  4314.5  906.89  4413.5  902.98  4441.8  900.82  4569.1   896.6  4639.8  893.09
 4710.34888.5576  4724.6  887.27  4795.4  886.11  4851.9  888.11  4866.1   887.5
  4929.3  887.34  4965.1  886.63  4979.2  884.91  4988.2  881.49  4989.2  880.69
  4997.5  880.69  4998.4  881.49  5035.8  883.27  5049.9  882.56  5064.1  884.01
  5106.5  885.82  5120.6  887.71 5136.89888.5578  5233.8   890.7    5402  892.68
    5559  895.23  5615.6  897.82  5643.9   900.4  5668.9  901.64  5728.7  904.48
#Mann= 6 ,-1 , 0
  4314.5      .1       0  4929.3     .16       0  4988.2     .07       0
  4998.4     .16       0    5402      .1       0  5668.9     .16       0
Bank Sta=4710.34,5136.89
XS Rating Curve= 0 ,0
Exp/Cntr=0.3,0.1

Type RM Length L Ch R = 1 ,146644  ,376,376,376
BEGIN DESCRIPTION:
CHACON CREEK 193.0
END DESCRIPTION:
XS GIS Cut Line= 3
      1989774.98     13672924.98        1989375.       13672425.
        1988875.       13672025.
#Sta/Elev= 30
    4369  902.82  4454.6  900.26  4539.5  896.01  4632.3  892.89 4689.92 886.895
  4710.7  885.38  4731.1  885.24  4789.2  884.33  4902.8  886.18  4923.6   884.6
  4931.6  882.15    4938   881.5  4952.5  882.85  4966.9  883.09  4981.3  882.78
  4982.6  881.46  4983.5  880.66  4991.8  880.66  4992.8  881.46  5002.1   882.5
  5012.5  882.54  5016.5  883.48  5051.7  882.77  5115.7  885.97  5243.8  886.19
 5279.96886.8952  5336.6  888.86  5414.4  890.33    5572  894.61  5649.6  898.42
#Mann= 5 ,-1 , 0
    4369      .1       0  4731.1     .16       0  4982.6     .07       0
  4992.8     .16       0  5414.4      .1       0
Bank Sta=4689.92,5279.96
XS Rating Curve= 0 ,0
Exp/Cntr=0.3,0.1

Type RM Length L Ch R = 1 ,146268  ,507,507,507
BEGIN DESCRIPTION:
CHACON CREEK 192.0
END DESCRIPTION:
XS GIS Cut Line= 3
      1989875.02     13672625.03        1989525.       13672125.
        1989075.       13671925.
#Sta/Elev= 30
  4355.8   897.1  4464.4  892.31  4485.3  890.51  4491.4  889.22  4506.2  888.15
  4527.2  885.36 4539.16884.6228  4563.3  883.64  4628.3  882.93  4771.3  884.08
  4866.3  883.89  4887.3  883.64  4909.2  881.91  4968.9  881.04  4980.5  879.97
  4982.9   878.4  4983.8   877.6  4992.2   877.6  4993.1   878.4  5009.9  879.49
  5020.9  879.28  5050.3  882.12  5064.7  882.74 5157.65884.6232  5195.3  885.93
  5351.2  888.02  5397.7  890.12    5421  892.33  5448.9  893.84  5458.6  894.28
#Mann= 5 ,-1 , 0
  4355.8      .1       0  4909.2     .16       0  4982.9     .07       0
  4993.1     .16       0  5448.9      .1       0
Bank Sta=4539.16,5157.65
XS Rating Curve= 0 ,0
Exp/Cntr=0.3,0.1

Type RM Length L Ch R = 1 ,145761  ,399,399,399
BEGIN DESCRIPTION:
CHACON CREEK 191.0
END DESCRIPTION:
XS GIS Cut Line= 3
      1990024.99     13672474.98        1989799.     13671794.72
      1989189.82     13671445.88
#Sta/Elev= 30
  3998.6  894.95    4125  892.45    4273  885.43  4362.7  883.81    4368  883.07
  4394.4  883.32  4399.7  882.24 4426.25881.9822  4526.3  880.36    4616  881.68
  4647.7  881.28  4679.4  880.08  4684.6  879.26  4731.5  878.77  4827.5  881.06
  4902.3  880.97  4924.4  880.25  4945.5  877.96  4982.9  876.88  4983.5  875.91
  4984.5  875.11  4992.9  875.11  4993.8  875.91 5020.82881.9819  5025.7  882.67
  5069.2  884.39  5238.6  885.95  5273.6  888.73  5305.2  890.18  5417.4  892.26
#Mann= 5 ,-1 , 0
  3998.6      .1       0  4924.4     .16       0  4983.5     .07       0
  4993.8     .16       0  5025.7      .1       0
Bank Sta=4426.25,5020.82
XS Rating Curve= 0 ,0
Exp/Cntr=0.3,0.1

Type RM Length L Ch R = 1 ,145362  ,780,780,780
BEGIN DESCRIPTION:
CHACON CREEK 190.0
END DESCRIPTION:
XS GIS Cut Line= 3
      1991132.33     13671815.56      1990075.04     13671508.27
      1989173.96     13671086.37
#Sta/Elev= 30
  3614.7  902.41  3903.5  895.41  3925.4  894.04  3958.9  894.27  4070.1  891.17
  4257.6  888.51  4382.2  883.54 4624.19880.4135  4726.8  879.32  4733.8  877.97
  4748.9   877.6    4771  878.14  4802.3  876.63  4815.2   874.4  4867.2  876.01
  4927.5  876.41  4967.6   878.4  4980.8  878.08  4990.5  876.86    4996  874.94
  5008.2   874.4  5009.1   873.6  5017.6   873.6  5018.5   874.4  5039.6   877.8
 5097.86880.4136  5366.9  886.62  5446.4   890.3    5555  893.76  5710.7  897.12
#Mann= 5 ,-1 , 0
  3614.7      .1       0  4867.2     .16       0  5008.2     .07       0
  5018.5     .16       0  5039.6      .1       0
Bank Sta=4624.19,5097.86
XS Rating Curve= 0 ,0
Exp/Cntr=0.3,0.1

Type RM Length L Ch R = 1 ,144582  ,494,494,494
BEGIN DESCRIPTION:
CHACON CREEK 189.0
END DESCRIPTION:
XS GIS Cut Line= 3
      1990974.96     13671274.98        1990175.       13670975.
      1989179.79     13670842.84
#Sta/Elev= 30
  4173.2  894.59  4243.5   893.8  4334.2  890.76  4353.8  891.22  4384.1  889.44
  4621.7  880.17  4693.4  878.84 4821.02877.5643  4896.7  876.81  4932.3  875.48
  4951.9  873.39  5001.4  872.54  5006.2  872.52  5007.1  871.46  5007.9  870.66
  5016.9  870.66  5017.8  871.46  5024.9  872.46  5137.5  876.31  5158.7  875.26
  5178.9  872.94  5209.1  875.09  5229.3  875.26 5252.22877.5643  5299.9  879.95
  5524.1  885.08  5670.7  890.43  5915.3  895.18    5979  897.33  6031.5  900.07
#Mann= 5 ,-1 , 0
  4173.2      .1       0  4693.4     .16       0  5001.4      .1       0
  5007.1     .07       0  5017.8      .1       0
Bank Sta=4821.02,5252.22
XS Rating Curve= 0 ,0
Exp/Cntr=0.3,0.1

Type RM Length L Ch R = 1 ,144088  ,709,709,709
BEGIN DESCRIPTION:
CHACON CREEK 188.0
END DESCRIPTION:
XS GIS Cut Line= 3
        1991325.       13670725.        1990125.       13670525.
      1989165.62     13670558.09
#Sta/Elev= 30
  3805.5  897.58  4038.7  891.68  4190.7  885.66  4203.4  886.37  4259.2  881.92
  4264.2  883.79  4302.3  881.06  4332.7  881.77  4380.8  880.16  4385.9  881.58
  4446.7  883.54  4507.6  883.37 4637.01875.7415  4707.8  872.58    4725  873.33
    4799  872.19  4806.6   873.5  4869.6   874.4  4933.3  873.75  4961.2  871.22
  4981.5  867.61  4996.4  867.39  4997.3  866.59  5007.1  867.39  5032.1  873.63
  5213.4875.7416  5372.3  879.94  5482.3  885.43  5782.5  893.79    5982  901.93
#Mann= 5 ,-1 , 0
  3805.5      .1       0    4725     .16       0  4869.6      .1       0
  4996.4     .07       0  5007.1      .1       0
Bank Sta=4637.01,5213.4
XS Rating Curve= 0 ,0
Exp/Cntr=0.3,0.1

Type RM Length L Ch R = 1 ,143379  ,424,424,424
BEGIN DESCRIPTION:
CHACON CREEK 187.0
END DESCRIPTION:
XS GIS Cut Line= 3
      1991144.78     13670287.25      1990353.16     13670155.31
       1989360.1     13670065.03
#Sta/Elev= 30
  4512.3  896.65  4633.7  892.74  4734.5   891.8  4916.9  888.08  4937.9  886.23
    4948  883.79  4958.1  879.61 4970.51872.6078  4977.8  868.84  4982.8   868.5
  4983.2  866.95    4984  866.15  4993.2  866.15    4994  866.95  5089.9  871.36
  5150.8  872.99  5226.2  871.19  5272.4  871.89  5302.8  870.86  5343.1  872.45
  5383.3  871.68  5413.4   872.8  5614.2   870.4  5654.4  871.68  5714.6  871.21
  5834.5872.6074  5865.3  873.31  5923.1  877.37  6038.6   882.1    6312  895.99
#Mann= 3 ,-1 , 0
  4512.3      .1       0  4983.2     .07       0    4994      .1       0
Bank Sta=4970.51,5834.5
XS Rating Curve= 0 ,0
Exp/Cntr=0.3,0.1

Type RM Length L Ch R = 1 ,142955  ,644,644,644
BEGIN DESCRIPTION:
Mapping XS 22f95d55
END DESCRIPTION:
XS GIS Cut Line= 4
      1991348.79     13670022.78      1990580.59      13669818.8
      1990098.82     13670061.85      1989249.08     13669966.47
#Sta/Elev= 30
  4134.8  898.69  4190.5  897.74  4219.9   895.5  4340.5  892.76    4531  885.66
  4542.2  886.04  4576.3  882.84  4645.7  882.48  4666.4  880.42  4718.1  879.26
  4759.5  876.32  4772.1  877.46 4825.57872.1254  4882.2  867.12  4929.6  866.94
  4992.8  864.64  4993.6  863.84  5003.6  864.64  5020.5  865.74  5026.1  867.25
  5081.5   866.5  5198.9  869.47  5361.5  870.64  5451.1  869.63  5722.5872.1254
  5757.3  873.27  5805.1  877.41  5847.4  878.31    6258  896.98  6324.3  898.68
#Mann= 3 ,-1 , 0
  4134.8      .1       0  4992.8     .07       0  5003.6      .1       0
Bank Sta=4825.57,5722.5
XS Rating Curve= 0 ,0
Exp/Cntr=0.3,0.1

Type RM Length L Ch R = 1 ,142311  ,41,41,41
BEGIN DESCRIPTION:
Mapping XS e3a879ce
END DESCRIPTION:
XS GIS Cut Line= 6
      1990962.53     13669918.62      1990298.48     13669653.87
      1990168.27     13669610.46      1990142.23     13669679.91
       1990020.7     13670031.47      1989313.21     13669957.68
#Sta/Elev= 30
  3809.6  885.96  4024.8   876.5    4049  877.56 4104.07872.0455  4186.5  873.08
  4239.4  868.85  4342.9  866.52  4396.8  866.45  4402.2  868.53  4450.7  866.52
  4456.1  868.44  4480.3  865.04  4485.7  867.54  4504.6  864.74    4510  867.57
  4535.1  863.72  4540.3  865.48  4605.8  863.68  4725.8  863.55  4775.8  870.19
  4838.2  871.54  4926.4  869.28  4988.8  870.88  5000.4  862.96  5001.2  862.16
  5011.2  862.96  5037.5  870.11 5289.95872.0449  5465.5  881.75  5819.2  896.01
#Mann= 6 ,-1 , 0
  3809.6      .1       0  4239.4     .05       0  4605.8     .16       0
  4725.8      .1       0  5000.4     .07       0  5011.2      .1       0
Bank Sta=4104.07,5289.95
XS Rating Curve= 0 ,0
Exp/Cntr=0.3,0.1

Type RM Length L Ch R = 1 ,142270  ,66,66,66
BEGIN DESCRIPTION:
Mapping XS 6db1c506
END DESCRIPTION:
XS GIS Cut Line= 6
      1991031.94     13669918.61       1990354.9     13669636.51
      1990155.25      13669571.4       1990107.5     13669623.48
      1989990.32     13669996.75      1989204.77     13669922.97
#Sta/Elev= 30
  3670.6  888.11  3970.6  877.26    4014  873.22  4167.1   873.6  4338.3  871.38
  4427.6  874.52  4454.3  873.12  4459.6  874.84  4486.2  871.83  4491.5  874.38
  4518.1  871.53  4523.4  874.17  4543.4  872.28  4638.5  875.19  4688.1  875.58
  4713.5  873.26  4718.6  875.25  4835.7  874.66 4887.75870.7999  4915.4  868.32
    4979  869.28  4994.8  864.36  4995.6  863.56  5005.6  864.36  5021.9  869.21
 5080.27870.7999  5232.3  872.18  5423.1  883.05  5784.7  896.83  5865.3  897.92
#Mann= 6 ,-1 , 0
  3670.6      .1       0  4167.1     .05       0  4543.4     .16       0
  4638.5      .1       0  4994.8     .07       0  5005.6      .1       0
Bank Sta=4887.75,5080.27
XS Rating Curve= 0 ,0
Exp/Cntr=0.3,0.1

Type RM Length L Ch R = 1 ,142204  ,378,378,378
BEGIN DESCRIPTION:
Mapping XS 6405e13b
END DESCRIPTION:
XS GIS Cut Line= 6
       1990984.2     13669844.83      1990229.03     13669567.06
      1990137.89     13669545.36      1990103.16     13669562.72
      1989920.87     13669979.39      1989197.99     13669884.16
#Sta/Elev= 30
  3688.6  884.85  3936.2  874.61  4115.5  874.31  4397.1  873.99  4402.4  871.82
  4452.7  872.86 4457.99870.5143  4483.1   872.9  4494.2  870.85  4523.4  873.32
  4528.5  870.58  4559.1  871.06  4590.1  865.43  4613.5  865.19  4614.3  864.39
  4624.3  865.19  4656.6   868.8  4662.1   866.1  4679.7  872.85  4685.2  869.34
  4702.8     873  4708.3  869.21  4725.8  871.08  4731.3  867.94  4869.1   870.8
  4999.6  865.83 5060.25870.5165  5167.2  872.42  5449.6  886.65  5809.7  896.33
#Mann= 6 ,-1 , 0
  3688.6      .1       0  4115.5     .05       0  4494.2     .16       0
  4590.1      .1       0  4613.5     .07       0  4624.3      .1       0
Bank Sta=4457.99,5060.25
XS Rating Curve= 0 ,0
Exp/Cntr=0.3,0.1

Type RM Length L Ch R = 1 ,141826  ,398,398,398
BEGIN DESCRIPTION:
Mapping XS f867484f
END DESCRIPTION:
XS GIS Cut Line= 4
      1990906.16     13669797.11      1990146.57     13669510.64
      1989803.69     13669627.83      1989070.18     13669397.79
#Sta/Elev= 30
  3981.3  880.36  4090.6   877.7  4121.5  875.08  4175.9  873.47  4319.3  872.47
  4346.4  872.92  4365.9  875.14  4371.2  873.69  4396.1  875.84  4401.4   874.2
  4420.7  874.72  4511.6  870.63  4627.3  870.83 4717.51868.9755  4808.1  865.31
  4889.9  864.93  4910.3  866.73  4946.9  865.43  4947.8  863.62  4948.6  862.82
  4958.7  863.62  4963.9  865.27    4985  863.96 5051.61868.9753  5072.1  869.18
  5129.5  876.01  5241.8  880.79  5483.3  890.64  5553.4   897.1  5924.2   913.6
#Mann= 7 ,-1 , 0
  3981.3      .1       0  4319.3     .05       0  4627.3     .16       0
  4808.1      .1       0  4947.8     .07       0  4958.7      .1       0
  5241.8     .16       0
Bank Sta=4717.51,5051.61
XS Rating Curve= 0 ,0
Exp/Cntr=0.3,0.1

Type RM Length L Ch R = 1 ,141428  ,557,557,557
BEGIN DESCRIPTION:
Mapping XS e66bc23f
END DESCRIPTION:
XS GIS Cut Line= 5
      1990939.95     13669790.14      1990468.62     13669615.67
      1990132.68     13669490.67      1989911.81       13668941.
       1989195.2     13668675.57
#Sta/Elev= 30
  3880.5  880.79  3981.7  877.33  4013.7  877.94  4113.2  872.66  4248.4  872.05
  4340.4  872.73  4424.4  870.91  4542.2  870.72 4699.47867.0552    4750  865.63
  4775.6  865.81    4877  863.76    4888  862.07  4912.2  863.91  4960.5  860.71
  4961.3  859.91  4971.4  860.71  4978.6  861.22  4990.1  862.06  4995.5  860.78
  5019.7  865.96  5081.7  865.41 5094.22867.0554  5127.2  874.77  5333.9  879.54
  5740.5   897.3  5856.7  904.65    5998  917.04  6045.4  919.26  6098.1   922.7
#Mann= 10 ,-1 , 0
  3880.5      .1       0  4248.4     .05       0  4424.4      .1       0
  4542.2     .16       0    4750      .1       0  4775.6     .16       0
  4960.5     .07       0  4971.4     .16       0  4978.6      .1       0
  6045.4     .16       0
Bank Sta=4699.47,5094.22
XS Rating Curve= 0 ,0
Exp/Cntr=0.3,0.1

Type RM Length L Ch R = 1 ,140871  ,124,124,124
BEGIN DESCRIPTION:
Mapping XS 66e06a5b
END DESCRIPTION:
XS GIS Cut Line= 6
      1991157.82     13669862.19      1990251.26     13669397.51
      1990367.05     13669002.54      1990450.39      13668856.7
      1990429.55     13668585.87      1990144.82     13668363.64
#Sta/Elev= 30
  3467.3  890.98  3751.4  879.72  3785.1  877.07  3807.6  878.11  3830.1  875.49
  3912.4  872.73    3929  873.16  3934.6  872.19  4444.3  869.14  4553.4  867.73
  4765.8  864.89 4789.06864.5103  4832.2  862.42  4837.4   863.2  4863.8  860.46
  4933.2   860.3  4966.8  860.19  4977.2  859.12    4978  858.32  4988.1  859.12
  5034.3  860.22  5068.1  861.41 5093.11  864.51  5107.4  866.27  5147.5   867.8
  5235.8  868.79  5368.8  869.77  5455.7  873.79  5590.4  877.56  5698.4  882.11
#Mann= 9 ,-1 , 0
  3467.3      .1       0  4444.3     .16       0  4553.4      .1       0
  4765.8     .16       0  4933.2      .1       0  4977.2     .07       0
  4988.1      .1       0  5034.3     .16       0  5235.8      .1       0
Bank Sta=4789.06,5093.11
XS Rating Curve= 0 ,0
Exp/Cntr=0.3,0.1

Type RM Length L Ch R = 1 ,140747  ,613,613,613
BEGIN DESCRIPTION:
Mapping XS 900697ed
END DESCRIPTION:
XS GIS Cut Line= 5
      1991353.15     13669780.31      1990367.05     13669335.87
      1990519.83      13669044.2      1990589.28     13668509.48
      1990130.91     13668287.24
#Sta/Elev= 30
  3446.5  894.63  3500.4  891.69  3587.1  889.29    3616  887.25  3835.3  879.85
  3863.9  877.01  3894.2  878.76  3910.1  876.29  3956.4  873.82  4031.3  872.93
  4100.7   870.6  4441.1  869.15  4837.9  865.63 4919.71863.9753  4934.3  861.85
  4939.3  862.67  4962.1   858.3  4962.9   857.5    4973   858.3  5038.1  859.83
  5078.4  859.25  5087.6  860.24  5092.6  859.43  5114.6  862.83 5125.45863.9753
    5149  866.28  5312.5  867.46  5553.6  870.64  5643.9   875.2    5906  883.51
#Mann= 5 ,-1 , 0
  3446.5      .1       0  4962.1     .07       0    4973      .1       0
  5114.6     .16       0  5312.5      .1       0
Bank Sta=4919.71,5125.45
XS Rating Curve= 0 ,0
Exp/Cntr=0.3,0.1

Type RM Length L Ch R = 1 ,140134  ,395,395,395
BEGIN DESCRIPTION:
CHACON CREEK 183.0
END DESCRIPTION:
XS GIS Cut Line= 3
        1991625.       13669225.        1991075.       13668625.
      1990314.55     13668082.26
#Sta/Elev= 30
  4206.6  888.46  4221.8  887.88  4284.6  884.03  4358.9  873.71  4425.8  866.22
  4482.5  864.62  4553.4   864.2  4666.9  861.83  4708.8  862.68  4808.1  862.92
  4885.8  862.63 4952.33861.4199  4970.9  858.93    4987  853.19  4987.8  852.39
  4997.2  852.39  4997.9  853.19  5006.7  855.26  5017.1  856.18  5070.9  856.38
  5093.1  858.33  5099.2  859.77  5120.1  860.74  5128.7   860.2  5134.8   860.8
 5272.38  861.42  5364.5  864.97  5535.4  869.33  5801.4   875.8  5954.8   879.7
#Mann= 8 ,-1 , 0
  4206.6      .1       0  4221.8     .16       0  4358.9      .1       0
    4987     .07       0  4997.9      .1       0  5070.9     .16       0
  5535.4      .1       0  5801.4     .16       0
Bank Sta=4952.33,5272.38
XS Rating Curve= 0 ,0
Exp/Cntr=0.3,0.1

Type RM Length L Ch R = 1 ,139739  ,438,438,438
BEGIN DESCRIPTION:
CHACON CREEK 182.0
END DESCRIPTION:
XS GIS Cut Line= 3
      1991861.37     13668759.31        1991425.       13668425.
      1990460.39     13667884.35
#Sta/Elev= 30
  4436.6  879.26  4483.3  877.77  4617.2  872.65  4668.5  870.94  4787.6  868.51
  4850.3  865.97 4930.02860.2893    4950  858.38  4958.2  856.55    4979  855.45
  4983.2  853.71  5010.5  853.18  5011.3  852.38  5020.7  852.38  5021.5  853.18
  5061.9  856.56  5089.5  857.98  5162.1   859.3  5227.1  858.49    5250  856.85
  5272.4  859.41  5412.7  858.59  5442.8  858.09  5480.8  860.29  5567.2  861.06
  5594.6   863.1  5794.3  868.99  5846.1  871.95  6039.5  876.32  6092.1  877.31
#Mann= 11 ,-1 , 0
  4436.6      .1       0  4483.3     .16       0  4617.2      .1       0
  4668.5     .16       0  4787.6      .1       0  5010.5     .07       0
  5021.5      .1       0  5061.9      .1       0  5272.4     .16       0
  5412.7      .1       0  6039.5     .16       0
Bank Sta=4930.02,5480.8
XS Rating Curve= 0 ,0
Exp/Cntr=0.3,0.1

Type RM Length L Ch R = 1 ,139301  ,508,508,508
BEGIN DESCRIPTION:
CHACON CREEK 181.0
END DESCRIPTION:
XS GIS Cut Line= 3
      1991975.02     13668575.03        1991675.       13668075.
      1990475.03     13667675.01
#Sta/Elev= 30
  4417.8  876.92  4542.2  871.61  4871.1  862.21  4934.8  861.27  4950.4  860.59
 4954.51859.0808  4965.9  857.67  4977.6  852.27  4987.7  851.17  4988.5  850.37
  4997.9  850.37  4998.7  851.17  5003.6  851.41  5011.5  854.19    5022  855.09
    5138  857.11  5190.7  856.87  5222.3  855.45  5253.9  856.91  5306.6  857.69
  5390.9  856.47  5490.1  857.08  5580.7  857.63 5612.13 859.079  5759.9  864.56
  5833.7   865.5  5928.5  871.14  5970.7  872.54  6097.2  874.96  6265.8  880.22
#Mann= 5 ,-1 , 0
  4417.8      .1       0  4871.1     .16       0  4987.7     .07       0
  4998.7     .16       0  5490.1      .1       0
Bank Sta=4954.51,5612.13
XS Rating Curve= 0 ,0
Exp/Cntr=0.3,0.1

Type RM Length L Ch R = 1 ,138793  ,490,490,490
BEGIN DESCRIPTION:
CHACON CREEK 180.0
END DESCRIPTION:
XS GIS Cut Line= 3
      1992752.06     13668097.89        1991475.       13667675.
      1990875.02     13667525.01
#Sta/Elev= 30
  3647.3  878.74    4184  867.31  4247.4  863.97  4273.9  859.88  4311.2857.2731
  4360.5  854.41  4385.3  854.74    4536  854.49  4560.5  855.37  4691.3  854.91
  4866.1  857.08    4945  854.76  4984.3  851.39    4985  850.59  4995.5  851.39
  5033.8  852.07    5075  854.86  5157.1  856.38  5281.2  855.81  5394.6  858.68
 5415.31857.2728  5422.9  858.85  5428.1  858.02  5464.1  864.04  5469.3   862.9
  5505.4  866.03  5510.5  864.23  5546.6  869.24  5551.8   867.9    5611  871.88
#Mann= 7 ,-1 , 0
  3647.3      .1       0  4385.3     .16       0    4536      .1       0
  4560.5     .16       0  4984.3     .07       0  4995.5     .16       0
  5157.1      .1       0
Bank Sta=4311.2,5415.31
XS Rating Curve= 0 ,0
Exp/Cntr=0.3,0.1

Type RM Length L Ch R = 1 ,138303  ,40,40,40
BEGIN DESCRIPTION:
Mapping XS 96f69788
END DESCRIPTION:
XS GIS Cut Line= 6
      1992663.52     13668009.35       1991606.2     13667621.31
      1991655.68     13667491.11      1991788.49     13667407.77
      1991806.72     13667329.65      1991351.79      13666929.3
#Sta/Elev= 30
  3519.3  875.75    4029  864.29 4094.03854.9442  4135.6  852.75  4379.2  854.09
  4625.6  856.65  4768.7  854.09  4774.4  855.99  4804.3  857.71  4819.5  855.96
  4825.4  852.87  4840.6  854.06  4846.6  851.88  4861.8  853.79  4867.7  851.61
    4877  852.92    4883  849.89  4896.7  851.66  4904.1  849.79  4974.1  849.32
  4974.8  848.52  4985.3  849.32  5023.1  849.44  5040.3  851.61 5046.79854.9435
  5061.2   857.9    5074  857.91  5210.1  860.21  5373.3  866.89  5634.5   872.1
#Mann= 5 ,-1 , 0
  3519.3      .1       0  4379.2     .16       0  4974.1     .07       0
  4985.3     .16       0    5074      .1       0
Bank Sta=4094.03,5046.79
XS Rating Curve= 0 ,0
Exp/Cntr=0.3,0.1

Type RM Length L Ch R = 1 ,138263  ,51,51,51
BEGIN DESCRIPTION:
CHACON CREEK 179.0
END DESCRIPTION:
XS GIS Cut Line= 6
      1992804.12     13668030.17      1991663.49     13667535.38
      1991843.18      13667423.4       1991856.2     13667368.71
      1991830.16       13667301.      1991374.44     13666899.97
#Sta/Elev= 30
  3457.3  878.23  3658.4  874.48  3892.4   867.4  4084.5   863.7  4136.9  860.21
 4175.66854.1944  4219.4  851.18  4411.4  852.99  4434.7  849.02  4435.4  848.22
  4445.9  849.02  4463.7  853.34  4487.3  853.22 4511.07854.1943  4685.8  856.17
  4697.1  858.51  4704.4  858.51  4709.7  856.78  4731.1  859.64    4832  862.21
    4982  862.25  4987.3  859.44    5012  862.34  5017.3  860.48  5036.4   862.8
  5067.7  862.85    5127  857.93  5226.9  859.66  5339.9  865.72  5648.8  871.91
#Mann= 5 ,-1 , 0
  3457.3      .1       0  4434.7     .07       0  4445.9      .1       0
  4487.3     .16       0  5067.7      .1       0
Bank Sta=4175.66,4511.07
XS Rating Curve= 0 ,0
Exp/Cntr=0.3,0.1

Type RM Length L Ch R = 1 ,138212  ,394,394,394
BEGIN DESCRIPTION:
Mapping XS 636e0477
END DESCRIPTION:
XS GIS Cut Line= 6
      1992772.84     13667941.62      1991754.64     13667535.38
      1991850.99     13667491.11      1991892.66     13667412.98
      1991903.08     13667332.25        1991443.     13666859.16
#Sta/Elev= 30
  3606.5  876.05  3796.2  871.86  3909.4  867.17  4149.2     862  4203.1  859.85
 4269.78 853.508  4325.5  849.96  4347.1  851.66  4424.1  851.28  4496.9   852.5
  4508.6  849.15  4519.3  848.89  4526.5  851.09  4540.9   852.9  4588.8  853.65
  4688.2  854.68  4836.4  853.42  4853.5  853.32  4945.7  852.35  4977.1  848.32
  4977.8  847.52  4987.6  847.52  4988.3  848.32  5018.1  852.84 5028.65853.5086
  5039.6  855.35  5066.2  856.76  5131.5  856.83  5393.1  865.75  5639.1  870.22
#Mann= 7 ,-1 , 0
  3606.5      .1       0  4588.8     .16       0  4836.4      .1       0
  4853.5     .16       0  4977.1     .07       0  4988.3     .16       0
  5066.2      .1       0
Bank Sta=4269.78,5028.65
XS Rating Curve= 0 ,0
Exp/Cntr=0.3,0.1

Type RM Length L Ch R = 1 ,137818  ,499,499,499
BEGIN DESCRIPTION:
Mapping XS e5dc93c5
END DESCRIPTION:
XS GIS Cut Line= 4
      1992848.39     13667759.33      1992334.49     13667466.89
       1992166.1     13667144.75      1991640.04     13666793.18
#Sta/Elev= 30
  4258.5  869.82  4477.6  865.25    4527  864.31  4644.6  858.37  4666.2   856.1
  4676.3  857.56  4688.1  857.18  4697.9  856.36 4712.15851.7035  4714.1  851.32
  4725.3   848.6  4741.1  847.75  4746.9  845.31  4784.4   847.6  4825.4  847.95
  4850.6  848.25  4963.6  848.16    4976  847.39  4985.3  844.99    4991  845.63
    4993  844.18  4993.7  843.38  5004.2  844.18  5051.6  850.46  5189.6  851.55
 5425.61851.7028  5494.5  852.35  5551.6  854.59  5659.7  862.71    5846  866.75
#Mann= 9 ,-1 , 0
  4258.5      .1       0  4477.6     .16       0  4714.1      .1       0
  4825.4     .16       0  4850.6      .1       0  4963.6     .16       0
    4993     .07       0  5004.2     .16       0  5189.6      .1       0
Bank Sta=4712.15,5425.61
XS Rating Curve= 0 ,0
Exp/Cntr=0.3,0.1

Type RM Length L Ch R = 1 ,137319  ,534,534,534
BEGIN DESCRIPTION:
CHACON CREEK 178.0
END DESCRIPTION:
XS GIS Cut Line= 3
      1993171.33     13667493.73      1992658.29     13667162.98
      1991770.27     13666774.96
#Sta/Elev= 30
  4410.6  867.86  4523.7  864.61  4572.8   864.4  4653.8  862.68  4768.6  858.17
  4826.1  856.43  4864.7   856.1    4935  854.69  4971.3   851.5 4973.47849.9626
  4977.3  847.25  4986.4  842.44  4995.4   841.2  4996.1   840.4  5006.2   840.4
  5006.8   841.2  5007.6  841.96    5020  843.88  5046.4  846.21  5090.1  845.64
  5117.1  846.29    5204  847.38  5319.3  849.99 5382.09849.9604  5559.3  850.14
  5780.4   851.5  5821.2  854.02  5886.7  860.83  5926.2  862.57  5990.1  864.02
#Mann= 5 ,-1 , 0
  4410.6      .1       0  4864.7     .16       0  4995.4     .07       0
  5006.8     .16       0  5117.1      .1       0
Bank Sta=4973.47,5382.09
XS Rating Curve= 0 ,0
Exp/Cntr=0.3,0.1

Type RM Length L Ch R = 1 ,136785  ,152,152,152
BEGIN DESCRIPTION:
CHACON CREEK 177.0
END DESCRIPTION:
XS GIS Cut Line= 4
      1993593.53     13667130.66      1992798.37     13666491.76
      1992600.45     13666894.54      1991824.97     13666624.99
#Sta/Elev= 30
  3781.4   869.1  3856.2  866.14  3984.2  863.79    4197  856.94  4296.2  854.83
  4432.2  853.35  4459.4  852.08    4517  851.89    4581  853.16  4659.4  852.38
 4700.44849.6185  4793.8  846.49  4949.9  847.69  4978.4  843.99    4984  841.32
  4988.8  841.21  4989.4  840.41  4999.6  840.41  5000.2  841.21  5096.4   843.1
  5158.3  842.93  5262.7  845.62  5308.9   845.5    5436   848.1  5573.7  849.62
 5798.15849.6182  5905.4   853.2  5998.7  861.35  6024.5  861.75  6071.2  864.04
#Mann= 3 ,-1 , 0
  3781.4      .1       0  4988.8     .07       0  5000.2      .1       0
Bank Sta=4700.44,5798.15
XS Rating Curve= 0 ,0
Exp/Cntr=0.3,0.1

Type RM Length L Ch R = 1 ,136633  ,591,591,591
BEGIN DESCRIPTION:
Mapping XS b31f6884
END DESCRIPTION:
XS GIS Cut Line= 5
      1993607.39     13667061.19      1992735.87      13666411.9
      1992531.01     13666703.56      1992531.01     13666804.26
      1991778.73     13666502.65
#Sta/Elev= 30
  3760.1  866.87  3837.9  864.43  3924.2  863.46  4180.7  855.88  4301.6  854.54
  4416.3  851.23  4595.7  852.35  4648.6849.5629  4745.8  846.21  4922.3  847.08
  4949.3  844.31    4958  844.96  4972.8  839.78  4973.2   837.3  4973.8   836.5
    4984   836.5  4984.7   837.3  4999.9  838.01  5014.7  842.04  5029.5   841.6
  5086.1  844.09  5315.7  845.41  5493.6  848.61  5644.5  848.31 5783.79 849.563
  5816.9  850.28  5902.2   858.8    5956  861.86  6039.4  864.12  6114.5  864.69
#Mann= 3 ,-1 , 0
  3760.1      .1       0  4973.2     .07       0  4984.7      .1       0
Bank Sta=4648.6,5783.79
XS Rating Curve= 0 ,0
Exp/Cntr=0.3,0.1

Type RM Length L Ch R = 1 ,136042  ,546,546,546
BEGIN DESCRIPTION:
CHACON CREEK 176.0
END DESCRIPTION:
XS GIS Cut Line= 3
      1993541.41     13666748.69        1992525.       13665975.
      1992174.97     13665824.99
#Sta/Elev= 30
  3712.4  861.06  3755.8   859.9  3776.6  858.55  3833.6  857.34  3911.8  854.16
 4186.71 849.482    4234  846.71  4311.1  845.61  4668.6  845.25  4753.8  846.36
  4903.5  845.41  4911.8  843.29  4918.1  843.21  4926.3  840.97  4965.3  839.61
  4998.7  839.22  5016.7  838.85  5017.3  838.05  5027.5  838.05  5028.2  838.85
  5044.2     843  5056.9  843.28  5098.6  842.16  5120.3  840.57  5142.1   840.9
  5163.9  844.44  5196.5  848.43 5200.49 849.483  5203.7  850.33  5370.6  858.13
#Mann= 5 ,-1 , 0
  3712.4      .1       0  4965.3     .05       0  4998.7      .1       0
  5016.7     .07       0  5028.2      .1       0
Bank Sta=4186.71,5200.49
XS Rating Curve= 0 ,0
Exp/Cntr=0.3,0.1

Type RM Length L Ch R = 1 ,135496  ,53,53,53
BEGIN DESCRIPTION:
CHACON CREEK 175.0
END DESCRIPTION:
XS GIS Cut Line= 4
      1993725.01     13666825.01      1992954.62     13666016.06
      1992753.23     13665477.87       1992500.8     13665138.99
#Sta/Elev= 30
  3428.4  865.16 4003.11849.4655  4185.3  844.96  4354.9   845.5  4701.4  843.66
  4717.5  839.33  4726.3  840.71  4731.7  839.22  4770.8  844.58  4802.9  845.16
  4811.8   844.9  4834.9  840.22  4872.4   839.7  4877.7  837.67  4895.9  838.34
  4927.6  838.59    4933  836.68  4957.9  838.99  4963.3  836.31  4982.9   837.3
  5012.7  836.09  5013.3  835.29  5024.3  836.09  5043.4  838.46  5046.1  837.59
  5073.7  837.16    5119  842.26 5232.12849.4653  5342.5  853.12  5542.7  866.42
#Mann= 5 ,-1 , 0
  3428.4      .1       0  4895.9     .05       0  5012.7    .033       0
  5024.3     .05       0  5046.1      .1       0
Bank Sta=4003.11,5232.12
XS Rating Curve= 0 ,0
Exp/Cntr=0.3,0.1

Type RM Length L Ch R = 1 ,135443  ,111,111,111
BEGIN DESCRIPTION:
CHACON CREEK 174.0
END DESCRIPTION:
XS GIS Cut Line= 4
      1993742.84     13666776.51      1992951.15     13665807.73
      1992791.42     13665450.09      1992574.98     13665074.97
#Sta/Elev= 30
  3487.8  864.02    4042  850.16  4176.2  845.31  4297.6  843.53    4619843.2071
  4624.9  843.11  4631.4  841.28  4633.3  836.19    4634  835.39  4644.3  835.39
  4644.9  836.19 4674.32 843.206  4688.8   843.5  4744.6  848.47  4767.8  849.25
    4791  849.86  4837.4  848.95  4842.9  850.12  4860.6  849.38  4866.1  850.23
  4932.5   850.4  5038.1  849.99  5147.9  849.29  5153.6  848.08  5169.4  849.04
  5175.2  848.19  5410.7  852.99    5448  854.88  5475.3  858.14  5563.7  864.67
#Mann= 5 ,-1 , 0
  3487.8      .1       0  4633.3    .033       0  4644.9      .1       0
  4932.5     .05       0  5038.1      .1       0
Bank Sta=4619,4674.32
XS Rating Curve= 0 ,0
Exp/Cntr=0.3,0.1

Type RM Length L Ch R = 1 ,135332  ,530,530,530
BEGIN DESCRIPTION:
CHACON CREEK 173.0
END DESCRIPTION:
XS GIS Cut Line= 3
      1993774.08     13666724.42      1993013.65     13665651.48
      1992665.27     13665004.16
#Sta/Elev= 30
    3535  863.73  3734.4  858.62  4093.7  851.99  4307.8     845 4562.84842.1857
    4661  841.72  4667.1  837.34  4674.2  836.52  4696.7  839.03  4710.9  842.29
  4788.9     842  4818.5  844.03  4839.4  841.92  4891.5  841.03  4926.2  838.05
  4964.3  837.99  4980.4   835.6  4981.1   834.8  4991.4   834.8    4992   835.6
  5046.3  838.12  5051.9   837.4  5073.8  839.92  5095.9  839.87 5137.04842.1858
  5259.6  848.13  5467.4  852.96  5533.1  858.25  5549.3  858.22  5585.2  860.55
#Mann= 3 ,-1 , 0
    3535      .1       0  4980.4     .07       0    4992      .1       0
Bank Sta=4562.84,5137.04
XS Rating Curve= 0 ,0
Exp/Cntr=0.3,0.1

Type RM Length L Ch R = 1 ,134802  ,514,514,514
BEGIN DESCRIPTION:
CHACON CREEK 172.0
END DESCRIPTION:
XS GIS Cut Line= 3
      1994206.34      13666324.2      1993859.13     13665859.81
      1992921.61     13664670.55
#Sta/Elev= 30
  3513.3  863.66  3877.6     855  3927.6  852.63  4027.7   851.8  4206.2  848.09
  4363.3  842.27  4384.1  842.86  4462.7  840.35 4579.19839.5208  4619.9  837.63
  4647.1  838.66  4690.4  838.59  4711.2   837.5  4748.2  838.43  4853.9  837.89
  4911.7  835.49  4912.3   834.4  4912.9   833.6  4923.3   833.6  4923.9   834.4
  4932.5  835.77  4982.2  835.73  5003.4  834.65  5017.4  837.94  5031.9  839.08
 5269.41839.5208  5331.8  840.43  5373.4  844.37  5516.1  853.65  5607.5  857.16
#Mann= 3 ,-1 , 0
  3513.3      .1       0  4912.3     .07       0  4923.9      .1       0
Bank Sta=4579.19,5269.41
XS Rating Curve= 0 ,0
Exp/Cntr=0.3,0.1

Type RM Length L Ch R = 1 ,134288  ,930,930,930
BEGIN DESCRIPTION:
CHACON CREEK 171.0
END DESCRIPTION:
XS GIS Cut Line= 3
      1994636.03     13666037.74      1994167.29     13665343.32
      1993148.65     13664324.67
#Sta/Elev= 30
  3486.7  871.04    3683  864.86  3871.4   860.1  4108.3  851.12  4326.9  846.87
  4388.6  843.79  4487.6  840.64  4657.3  839.06 4683.31837.3006  4713.9  832.68
    4728  831.81  4749.2   834.1  4876.5  835.96  4918.9  835.31  4954.3  832.34
  4989.6  832.22    4998  830.84  4998.6  830.04    5009  830.04  5009.6  830.84
  5010.8  832.93  5017.9  834.61  5046.2  836.28  5180.6  835.47    5230  835.96
 5248.29837.3005  5265.4   838.5  5357.3  840.96  5562.4  844.84  5765.1  853.36
#Mann= 3 ,-1 , 0
  3486.7      .1       0    4998     .07       0  5009.6      .1       0
Bank Sta=4683.31,5248.29
XS Rating Curve= 0 ,0
Exp/Cntr=0.3,0.1

Type RM Length L Ch R = 1 ,133358  ,1370,1370,1370
BEGIN DESCRIPTION:
CHACON CREEK 170.0
END DESCRIPTION:
XS GIS Cut Line= 3
      1994921.61     13665331.13      1994374.76     13664357.21
      1993525.75     13663935.31
#Sta/Elev= 30
  4090.7  857.05  4120.7   857.3  4179.5  854.43  4246.8  852.19  4282.5  849.14
  4379.3  841.16    4482  835.37  4613.8  832.86 4692.26832.6698    4790  833.44
  4900.5  832.18  4957.9  830.49  4989.5  826.78  4990.1  825.98  5000.7  825.98
  5001.2  826.78  5048.9  831.07  5092.3  830.46  5157.3  831.69  5200.7  830.77
    5206  829.52    5224   829.1  5240.8  829.45  5246.4  831.26 5265.85832.6695
  5313.6   835.7  5358.4  836.97  5991.2  840.43  6058.5   841.8  6155.7  847.02
#Mann= 5 ,-1 , 0
  4090.7      .1       0  4179.5     .05       0  4282.5      .1       0
  4989.5     .07       0  5001.2      .1       0
Bank Sta=4692.26,5265.85
XS Rating Curve= 0 ,0
Exp/Cntr=0.3,0.1

Type RM Length L Ch R = 1 ,131988  ,42,42,42
BEGIN DESCRIPTION:
CHACON CREEK 168.0
END DESCRIPTION:
XS GIS Cut Line= 6
      1995837.42     13664399.71      1995656.88     13663896.27
      1995285.78     13663957.04      1994953.75       13664352.
      1994556.18     13663923.18      1993545.74     13663615.88
#Sta/Elev= 30
    4223  839.14  4367.4  840.17  4454.4  839.89  4808.5  837.05  4839.7  837.61
  4849.7  836.29  4884.2   834.3    4896832.1874  4919.8  826.98  5000.9  826.47
  5001.4  825.67    5012  825.67  5012.6  826.47    5452  826.47  5602.8  828.87
  5630.8  828.58  5752.7   830.2  5896.3  829.18  6188.8  831.09  6246.3  830.43
  6487.7  830.63 6521.71832.1874  6552.8  834.07  6585.6  832.58  6689.5  835.87
  6755.2  836.81  7061.4  838.35  7156.7  839.77  7261.2  843.47  7354.5  848.99
#Mann= 5 ,-1 , 0
    4223      .1       0  4808.5     .08       0  4884.2      .1       0
  5000.9     .07       0  5012.6      .1       0
Bank Sta=4896,6521.71
XS Rating Curve= 0 ,0
Exp/Cntr=0.3,0.1

Type RM Length L Ch R = 1 ,131946  ,65,65,65
BEGIN DESCRIPTION:
CHACON CREEK 169.0
END DESCRIPTION:
XS GIS Cut Line= 6
      1995876.49     13664409.28      1995741.08     13663867.63
      1995348.72     13663878.04      1994970.24     13664287.76
      1994645.59     13663878.04      1993524.98     13663524.99
#Sta/Elev= 30
  4109.9  838.62  4385.8  839.49  4818.7  835.25  4860.7  834.04  4955.9  834.54
    4961  832.22  5007.2  834.42  5123.8  834.39  5129.6  832.49  5145.2  834.26
    5151  832.41  5160.7  833.78 5166.06831.5806  5182.1  834.43  5187.9  833.04
  5203.5  834.69  5426.6   834.6  5524.6  836.33  5689.2  835.51  5727.8  833.61
  6146.3  834.16  6192.1  830.51  6271.9  829.58  6272.5  828.78  6283.6  829.58
 6551.25831.5792  6602.8  834.31  6707.7  835.89  7106.1  839.16  7368.2  851.63
#Mann= 5 ,-1 , 0
  4109.9      .1       0  4818.7     .08       0  4860.7      .1       0
  6271.9     .07       0  6283.6      .1       0
Bank Sta=5166.06,6551.25
XS Rating Curve= 0 ,0
Exp/Cntr=0.3,0.1

Type RM Length L Ch R = 1 ,131881  ,82,82,82
BEGIN DESCRIPTION:
CHACON CREEK 167.0
END DESCRIPTION:
XS GIS Cut Line= 6
      1995956.34     13664401.87      1995787.08     13663813.37
      1995354.79     13663808.16        1994985.     13664211.81
      1994693.33     13663825.09      1993569.19      13663481.6
#Sta/Elev= 30
  4002.2  836.92  4170.2  838.93    4488  837.45  4508.8  838.18  4611.1  835.08
    4717   834.6  4807.4  832.09 4939.82825.5656  4973.5   822.4  4978.5  823.05
  5032.8   820.4  5033.3   819.6  5043.9   819.6  5044.5   820.4    5137  823.91
  5245.5  824.14 5310.93825.5651  5345.7  825.88  5399.2  828.83    5434  827.76
  5595.6   829.8  5732.7  828.49  5861.6  830.36  6113.6  829.23  6475.9  830.25
  6541.5  833.17  6606.3  834.75  7059.5  838.83  7195.9  844.37    7292  850.21
#Mann= 3 ,-1 , 0
  4002.2      .1       0  5032.8     .07       0  5044.5      .1       0
Bank Sta=4939.82,5310.93
XS Rating Curve= 0 ,0
Exp/Cntr=0.3,0.1

Type RM Length L Ch R = 1 ,131799  ,818,818,818
BEGIN DESCRIPTION:
CHACON CREEK 166.0
END DESCRIPTION:
XS GIS Cut Line= 6
      1996526.67     13664734.22      1996011.04     13663781.08
      1995276.67     13663739.41      1995057.92     13663968.58
       1994922.5     13663775.87      1993709.49     13663338.56
#Sta/Elev= 30
  3284.9  840.66  3390.4  839.26  3504.3  837.39  3884.1  833.87  4037.3  828.87
  4222.9  828.65  4228.5  830.53    4239  830.33  4244.7  832.27  4266.6  832.62
  4406.8  829.08  4503.2  831.04  4688.4   831.1  4850.4  826.91  4923.4   826.4
  4960.7823.2745  4981.2  820.72  5026.7  820.16  5027.3  819.36  5038.5  820.16
 5114.51 823.275  5350.4  824.93  5371.5  827.95  5385.7  828.24    5407   826.2
  5506.1  827.68  6031.8  827.65    6395  834.51  6788.3  838.64  6953.6  844.28
#Mann= 7 ,-1 , 0
  3284.9      .1       0  3390.4     .08       0  3504.3      .1       0
  4222.9     .05       0  4406.8      .1       0  5026.7     .07       0
  5038.5      .1       0
Bank Sta=4960.7,5114.51
XS Rating Curve= 0 ,0
Exp/Cntr=0.3,0.1

Type RM Length L Ch R = 1 ,130981  ,19,19,19
BEGIN DESCRIPTION:
Mapping XS 0049a962
END DESCRIPTION:
XS GIS Cut Line= 6
      1996508.45     13664512.01      1996136.04     13663840.11
       1995357.4     13663342.71       1995419.9     13662972.92
      1995274.06     13663233.34      1994162.69     13662249.48
#Sta/Elev= 30
  2917.1  838.51  3382.4  835.51  3622.5  826.45  3754.4  828.31  3792.2   830.7
  3879.4  827.96 4489.47823.1165  4579.8  823.79  4607.7  818.79  4701.4  821.46
  4909.7  816.98  4914.8   819.3  4938.9  814.17  4973.3  813.67  4973.8  812.87
  4985.4  813.67  5141.2  814.15    5260  821.11    5322  818.15  5540.6  827.35
 5612.33823.1169  5699.3   830.5    5912  829.18  6026.1  836.86    6101  838.04
  6138.4  838.18  6257.2  838.93  6263.2   839.1  6391.9   840.8  6811.1  847.58
#Mann= 10 ,-1 , 0
  2917.1      .1       0  3754.4     .05       0  3879.4      .1       0
  4973.3     .07       0  4985.4      .1       0    6101     .08       0
  6138.4      .1       0  6257.2     .08       0  6263.2     .05       0
  6391.9      .1       0
Bank Sta=4489.47,5612.33
XS Rating Curve= 0 ,0
Exp/Cntr=0.3,0.1

Type RM Length L Ch R = 1 ,130962  ,24,24,24
BEGIN DESCRIPTION:
Mapping XS 30367260
END DESCRIPTION:
XS GIS Cut Line= 6
      1996531.88     13664499.84       1996172.5     13663833.16
      1995401.67     13663338.37      1995391.25      13662916.5
      1995266.25     13663187.33      1994194.31     13662209.06
#Sta/Elev= 30
  2920.9  838.73  3387.5  835.75  3674.4  825.83  3791.7  828.01  3916.6  827.53
 4508.59823.0107  4608.2  822.33  4668.3  826.46  4674.7  826.68  4817.3  827.69
  4837.9  820.87  4909.7     821  4948.8  813.89  5013.5  813.68    5014  812.88
  5025.7  813.68  5090.2  828.12 5426.26823.0106  5570.4  824.49  5712.3   831.4
  5775.8  827.54  5917.7  829.21  6076.6  837.74  6180.5  837.74    6228  838.69
  6289.5  838.97  6439.6  840.58    6682   844.3  6698.6  844.64  6828.2  847.31
#Mann= 14 ,-1 , 0
  2920.9      .1       0  3791.7     .05       0  3916.6      .1       0
  4668.3     .08       0  4674.7      .1       0  5013.5     .07       0
  5025.7      .1       0  6076.6     .08       0  6180.5      .1       0
    6228     .08       0  6289.5     .05       0  6439.6      .1       0
    6682     .05       0  6698.6      .1       0
Bank Sta=4508.59,5426.26
XS Rating Curve= 0 ,0
Exp/Cntr=0.3,0.1
