--- UNT 043 in HW.prj (project) ---

Proj Title=UNT 043 in HW Base Level Engineering
Current Plan=p01
Default Exp/Contr=0.3,0.1
English Units
Geom File=g01
Flow File=f01
Plan File=p01
Y Axis Title=Elevation
X Axis Title(PF)=Main Channel Distance
X Axis Title(XS)=Station
BEGIN DESCRIPTION:
UNT 043 in HW
END DESCRIPTION:
DSS Export Rating Curves= 0
DSS Export Rating Curve Sorted= 0
DSS Export Volume Flow Curves= 0
DXF OffsetX= 0
DXF OffsetY= 0
DXF ScaleX= 1
DXF ScaleY= 10

--- UNT 043 in HW.p01 (plan) ---

Plan Title=Multiple Run
Short Identifier=Multiple
Geom File=g01
Flow File=f01
Subcritical Flow
K Sum by GR= 0
Std Step Tol= 0.01
Critical Tol= 0.01
Num of Std Step Trials= 20
Max Error Tol= 0.3
Flow Tol Ratio= 0.001
Split Flow NTrial= 30
Split Flow Tol= 0.02
Split Flow Ratio= 0.02
Log Output Level= 0
Friction Slope Method= 1
Unsteady Friction Slope Method= 2
Unsteady Bridges Friction Slope Method= 1
Parabolic Critical Depth
Global Vel Dist=  1 , 1 , 1
Global Log Level= 0
CheckData=True
Encroach Param= -1, 0, 0, 0
BEGIN DESCRIPTION:
Multiple Run
END DESCRIPTION:

--- UNT 043 in HW.f01 (steady flow) ---

Flow Title=Multiple
Program Version=5.05
Number of Profiles= 7
Profile Names=10-year,25-year,50-year,1pct_min,100-year,1pct_plu,500-year
River Rch & RM=UNT 043 in HW,Reach-1         ,15278
     388     536     658     401     799    1595    1184
River Rch & RM=UNT 043 in HW,Reach-1         ,13539
     699     999    1253     779    1554    3101    2398
River Rch & RM=UNT 043 in HW,Reach-1         ,7697
    1052    1534    1952    1228    2449    4887    3874
River Rch & RM=UNT 043 in HW,Reach-1         ,2848
    1224    1798    2297    1450    2894    5774    4614
River Rch & RM=UNT 043 in HW,Reach-1         ,2427
    1224    1798    2297    1450    2894    5774    4614
Boundary for River Rch & Prof#=UNT 043 in HW,Reach-1         , 1
Up Type= 0
Dn Type= 3
Dn Slope=0.005
Boundary for River Rch & Prof#=UNT 043 in HW,Reach-1         , 2
Up Type= 0
Dn Type= 3
Dn Slope=0.005
Boundary for River Rch & Prof#=UNT 043 in HW,Reach-1         , 3
Up Type= 0
Dn Type= 3
Dn Slope=0.005
Boundary for River Rch & Prof#=UNT 043 in HW,Reach-1         , 4
Up Type= 0
Dn Type= 3
Dn Slope=0.005
Boundary for River Rch & Prof#=UNT 043 in HW,Reach-1         , 5
Up Type= 0
Dn Type= 3
Dn Slope=0.005
Boundary for River Rch & Prof#=UNT 043 in HW,Reach-1         , 6
Up Type= 0
Dn Type= 3
Dn Slope=0.005
Boundary for River Rch & Prof#=UNT 043 in HW,Reach-1         , 7
Up Type= 0
Dn Type= 3
Dn Slope=0.005
DSS Import GetInterval= 0
DSS Import GetPeak= 0
DSS Import FillOption= 0

--- UNT 043 in HW.g01 (geometry) ---

Geom Title=Existing Conditions

River Reach=UNT 043 in HW,Reach-1
Reach XY= 30
      1981708.38     13632156.96      1982630.80     13632064.54
      1983390.80     13632324.54      1983480.80     13632254.54
      1983550.80     13632014.54      1983480.80     13631134.54
      1983640.80     13630504.54      1984000.80     13630384.54
      1984240.80     13630174.54      1984500.80     13629604.54
      1984274.63     13629104.62      1984556.71     13628703.33
      1985033.79     13628467.91      1984871.29     13628203.33
      1984790.80     13627774.54      1984840.80     13627514.54
      1985070.80     13627374.54      1984920.80     13626854.54
      1985080.80     13626704.54      1985530.80     13626694.54
      1985660.80     13625614.54      1985810.80     13625434.54
      1986260.80     13625194.54      1987270.80     13624964.54
      1987680.80     13624964.54      1987860.80     13624834.54
      1987720.80     13624378.53      1988030.93     13623840.34
      1988040.80     13623324.54      1988360.80     13623184.54

Type RM Length L Ch R = 1,15278,165,165,165
BEGIN DESCRIPTION:
UNT 043 in HW 32.0
END DESCRIPTION:
XS GIS Cut Line= 3
      1981929.17     13632584.78      1981918.75     13632116.04
      1981811.11     13631640.33
#Sta/Elev= 30
  4529.6  808.57  4689.4  806.18  4749.4  804.77  4789.4  804.58  4809.5  803.29
  4829.5  804.18  4849.5  803.60  4881.2  803.39  4909.5  802.99  4941.2  803.76
  4979.5  803.90  4993.5  802.67  4994.0  801.87  4999.0  801.87  4999.5  802.67
  5001.6  802.67  5009.8  804.05  5102.1  803.29  5163.6  804.51  5194.3  804.68
  5214.5  805.31  5225.1  806.31  5255.8  806.72  5262.8  806.93  5267.9  807.58
  5306.0  807.74  5311.1  808.23  5348.1  809.05  5359.4  809.76  5486.2  811.61
#Mann=5,-1,0
  4529.6     0.1       0  4881.2    0.05       0  4941.2     0.1       0
  4993.5    0.07       0  4999.5     0.1       0
Bank Sta=4993.5,4999.5
Exp/Cntr=0.3,0.1

Type RM Length L Ch R = 1,15113,145,145,145
BEGIN DESCRIPTION:
Mapping XS 3ca28b15
END DESCRIPTION:
XS GIS Cut Line= 4
      1982045.36     13632606.02      1982092.24     13632167.21
      1982040.16     13631904.18      1981930.78     13631643.76
#Sta/Elev= 30
  4494.8  806.81  4534.7  806.78  4616.5  805.78  4676.9  804.49  4816.7  803.27
  4837.8  801.82  4867.9  802.29  4876.3  802.08  4934.7  801.44  4979.1  801.89
  4989.3  801.38  4993.8  800.52  4994.3  799.72  4999.3  799.72  4999.8  800.52
  5019.9  802.20  5061.0  802.42  5104.3  802.54  5225.1  801.82  5254.2  802.06
  5301.0  802.72  5307.2  803.07  5312.6  804.11  5322.7  804.46  5330.9  804.08
  5376.9  804.88  5442.2  806.82  5460.6  806.99  5466.0  807.49  5486.7  807.57
#Mann=5,-1,0
  4494.8     0.1       0  4876.3    0.05       0  4993.8   0.035       0
  4999.8    0.05       0  5061.0     0.1       0
Bank Sta=4993.8,4999.8
Exp/Cntr=0.3,0.1

Type RM Length L Ch R = 1,14968,148,148,148
BEGIN DESCRIPTION:
UNT 043 in HW 31.0
END DESCRIPTION:
XS GIS Cut Line= 4
      1982116.66     13632508.45      1982225.00     13632077.60
      1982170.77     13631722.10      1981972.46     13631491.00
#Sta/Elev= 30
  4573.2  805.32  4823.1  802.17  4833.5  801.82  4865.5  800.14  4872.3  800.48
  4886.1  800.30  4906.7  799.53  4959.7  798.64  4978.9  798.84  4989.2  797.82
  4995.7  797.59  4997.8  797.10  4998.3  796.30  5003.3  796.30  5003.8  797.10
  5016.2  798.98  5030.2  798.87  5048.0  797.63  5080.8  798.24  5180.1  799.16
  5323.6  799.22  5393.3  799.72  5471.2  801.76  5485.5  801.81  5492.1  802.35
  5499.8  802.23  5506.4  802.74  5542.6  802.64  5641.4  805.33  5681.6  805.62
#Mann=5,-1,0
  4573.2     0.1       0  4823.1    0.05       0  4833.5     0.1       0
  4997.8    0.07       0  5003.8     0.1       0
Bank Sta=4997.8,5003.8
Exp/Cntr=0.3,0.1

Type RM Length L Ch R = 1,14820,98,98,98
BEGIN DESCRIPTION:
Mapping XS c0220f10
END DESCRIPTION:
XS GIS Cut Line= 4
      1982325.74     13632394.68      1982367.41     13631964.95
      1982330.96     13631722.76      1982019.22     13631465.58
#Sta/Elev= 30
  4688.4  801.09  4858.9  799.68  4899.1  798.44  4919.2  798.47  4937.0  797.71
  4942.0  797.89  4969.4  796.60  4979.4  796.57  4996.5  794.78  4997.0  793.98
  5002.0  793.98  5002.5  794.78  5019.6  796.66  5029.7  796.88  5059.8  795.89
  5300.7  797.53  5374.3  798.64  5424.6  798.66  5474.7  799.43  5481.2  799.24
  5509.9  799.98  5573.7  799.72  5637.5  800.90  5651.9  801.74  5687.0  802.39
  5694.9  803.14  5722.8  802.62  5744.4  803.43  5750.9  803.25  5769.2  804.20
#Mann=3,-1,0
  4688.4     0.1       0  4996.5    0.07       0  5002.5     0.1       0
Bank Sta=4996.5,5002.5
Exp/Cntr=0.3,0.1

Type RM Length L Ch R = 1,14722,157,157,157
BEGIN DESCRIPTION:
Mapping XS a1bd92af
END DESCRIPTION:
XS GIS Cut Line= 3
      1982420.49     13632567.45      1982472.45     13631701.06
      1982039.23     13631344.08
#Sta/Elev= 30
  4506.2  799.11  4664.5  800.08  4769.1  799.02  4833.2  797.86  4909.4  797.41
  4959.5  796.44  4998.9  793.62  4999.4  792.82  5004.4  792.82  5004.9  793.62
  5009.6  794.19  5029.6  795.18  5049.6  794.61  5170.5  795.31  5290.1  797.21
  5376.6  796.79  5405.3  797.34  5440.4  797.33  5469.1  798.26  5497.8  798.47
  5596.8  797.58  5675.0  797.94  5689.3  798.64  5718.0  799.10  5817.0  799.43
  5831.3  800.19  5880.8  800.71  5909.5  801.97  5930.3  801.67  5935.5  802.16
#Mann=3,-1,0
  4506.2     0.1       0  4998.9    0.07       0  5004.9     0.1       0
Bank Sta=4998.9,5004.9
Exp/Cntr=0.3,0.1

Type RM Length L Ch R = 1,14565,248,248,248
BEGIN DESCRIPTION:
Mapping XS 709721d9
END DESCRIPTION:
XS GIS Cut Line= 3
      1982549.71     13632423.24      1982651.27     13631735.78
      1982104.41     13631303.50
#Sta/Elev= 30
  4637.4  796.95  4676.1  796.84  4709.6  796.09  4726.6  796.47  4756.9  795.95
  4774.2  796.29  4797.4  795.66  4837.8  795.95  4858.0  795.12  4918.7  794.32
  4949.0  794.63  4969.2  793.95  4996.5  791.58  4997.0  790.78  5002.0  790.78
  5002.5  791.58  5009.6  792.50  5029.9  793.76  5052.5  793.43  5186.7  795.20
  5332.3  794.73  5480.5  796.54  5571.8  796.11  5635.9  796.42  5708.1  797.51
  5813.8  796.62  5892.4  797.48  5921.2  798.60  5970.9  798.50  6029.4  799.53
#Mann=3,-1,0
  4637.4     0.1       0  4996.5    0.07       0  5002.5     0.1       0
Bank Sta=4996.5,5002.5
Exp/Cntr=0.3,0.1

Type RM Length L Ch R = 1,14317,377,377,377
BEGIN DESCRIPTION:
Mapping XS 32008f9f
END DESCRIPTION:
XS GIS Cut Line= 4
      1982533.23     13632571.36      1982814.50     13632222.38
      1982809.29     13631998.42      1982737.00     13631848.69
#Sta/Elev= 30
  4486.1  796.69  4556.3  796.13  4577.2  795.59  4591.5  795.74  4676.3  794.50
  4698.7  794.59  4725.9  793.74  4748.3  793.92  4783.5  793.57  4882.7  791.71
  4911.4  791.53  4925.8  791.94  4934.3  791.77  4951.7  792.05  4961.7  791.76
  4981.7  789.49  4988.7  789.32  4989.2  788.52  4994.2  788.52  4994.7  789.32
  5021.7  791.33  5031.7  791.68  5127.2  792.06  5132.2  792.42  5179.2  792.63
  5184.8  793.00  5201.8  793.00  5207.4  793.35  5230.0  793.65  5324.6  794.31
#Mann=3,-1,0
  4486.1     0.1       0  4988.7    0.07       0  4994.7     0.1       0
Bank Sta=4988.7,4994.7
Exp/Cntr=0.3,0.1

Type RM Length L Ch R = 1,13940,401,401,401
BEGIN DESCRIPTION:
Mapping XS f8991a2d
END DESCRIPTION:
XS GIS Cut Line= 4
      1982496.76     13632633.85      1982996.79     13632435.92
      1983179.08     13632159.88      1982840.57     13631904.70
#Sta/Elev= 30
  4208.9  797.79  4245.6  796.51  4383.4  793.96  4407.8  793.00  4454.4  791.99
  4486.2  791.49  4491.5  791.77  4529.7  790.89  4545.6  791.07  4594.2  789.56
  4624.0  789.63  4629.4  790.01  4707.8  788.51  4753.1  787.99  4768.2  788.57
  4825.4  787.58  4969.9  788.27  4984.9  787.20  4996.4  785.71  4996.9  784.91
  5001.9  784.91  5002.4  785.71  5006.0  786.51  5035.4  787.97  5063.2  787.31
  5162.2  788.03  5276.7  789.55  5333.1  790.70  5397.4  790.77  5501.4  792.15
#Mann=3,-1,0
  4208.9     0.1       0  4996.4    0.07       0  5002.4     0.1       0
Bank Sta=4996.4,5002.4
Exp/Cntr=0.3,0.1

Type RM Length L Ch R = 1,13539,264,264,264
BEGIN DESCRIPTION:
Mapping XS d33ad29c
END DESCRIPTION:
XS GIS Cut Line= 3
      1983882.21     13632540.09      1983028.04     13631967.17
      1982898.96     13631920.71
#Sta/Elev= 30
  4504.9  818.94  4542.3  815.53  4557.3  813.03  4564.5  812.62  4658.1  807.19
  4707.4  802.94  4716.4  804.09  4722.4  802.97  4743.4  801.07  4752.4  801.08
  4794.4  798.42  4845.4  796.08  4866.4  794.23  4881.4  794.33  4887.5  793.44
  4896.4  793.44  4902.5  792.39  4917.5  791.54  4968.5  784.48  4992.5  783.23
  4993.0  782.43  4998.0  782.43  4998.5  783.23  5031.5  785.21  5046.5  784.54
  5169.6  784.92  5292.6  787.23  5493.7  788.71  5579.0  790.65  5670.6  791.44
#Mann=4,-1,0
  4504.9    0.16       0  4564.5     0.1       0  4992.5    0.07       0
  4998.5     0.1       0
Bank Sta=4992.5,4998.5
Exp/Cntr=0.3,0.1

Type RM Length L Ch R = 1,13275,315,315,315
BEGIN DESCRIPTION:
Mapping XS f3e10941
END DESCRIPTION:
XS GIS Cut Line= 2
      1984095.70     13632149.45      1982850.92     13631878.62
#Sta/Elev= 30
  4428.6  829.62  4480.5  825.15  4567.3  819.23  4654.5  812.61  4660.4  811.67
  4683.7  809.95  4715.9  807.83  4758.6  805.97  4787.5  803.43  4818.2  802.04
  4846.6  797.34  4851.7  797.20  4895.7  790.60  4900.8  790.45  4930.8  786.66
  4951.2  782.97  4971.7  781.68  4990.9  781.09  4991.4  780.29  4996.4  780.29
  4996.9  781.09  5002.4  781.78  5022.9  782.64  5180.1  784.07  5273.2  785.58
  5350.4  787.61  5415.3  787.70  5508.4  789.07  5565.3  790.61  5702.5  792.15
#Mann=4,-1,0
  4428.6    0.16       0  4683.7     0.1       0  4990.9    0.07       0
  4996.9     0.1       0
Bank Sta=4990.9,4996.9
Exp/Cntr=0.3,0.1

Type RM Length L Ch R = 1,12960,305,305,305
BEGIN DESCRIPTION:
UNT 043 in HW 30.0
END DESCRIPTION:
XS GIS Cut Line= 3
      1984116.57     13631863.00      1983525.00     13631725.00
      1982725.96     13631743.21
#Sta/Elev= 30
  4398.5  818.22  4401.9  818.22  4408.5  816.75  4413.6  817.46  4451.0  812.92
  4456.2  813.81  4472.0  811.47  4490.7  810.30  4500.7  808.54  4589.7  801.04
  4605.5  799.62  4674.0  796.03  4721.7  792.28  4739.0  791.92  4764.3  789.96
  4790.3  789.46  4811.9  786.93  4903.3  782.23  4954.6  780.51  4992.7  777.93
  4993.2  777.13  4998.2  777.13  4998.7  777.93  5008.5  778.10  5026.0  780.03
  5136.0  782.94  5336.0  785.58  5566.1  791.22  5606.1  791.27  5805.2  794.29
#Mann=6,-1,0
  4398.5    0.16       0  4490.7     0.1       0  4500.7    0.16       0
  4589.7     0.1       0  4992.7    0.07       0  4998.7     0.1       0
Bank Sta=4992.7,4998.7
Exp/Cntr=0.3,0.1

Type RM Length L Ch R = 1,12655,271,271,271
BEGIN DESCRIPTION:
UNT 043 in HW 29.0
END DESCRIPTION:
XS GIS Cut Line= 3
      1984041.09     13631558.85      1983525.00     13631425.00
      1982764.98     13631522.39
#Sta/Elev= 30
  4462.6  807.42  4489.6  805.78  4510.2  803.32  4536.9  801.28  4653.4  796.96
  4665.2  796.02  4690.0  795.50  4727.2  794.97  4758.2  792.41  4809.8  786.16
  4815.7  784.78  4820.9  784.71  4856.3  779.32  4861.5  779.53  4902.8  776.97
  4932.3  777.29  4937.5  776.69  4985.4  776.33  4990.2  775.79  4990.7  774.99
  4995.7  774.99  4996.2  775.79  5076.4  779.41  5167.2  782.19  5257.9  783.15
  5368.8  786.71  5499.9  788.42  5585.7  790.66  5641.0  790.59  5762.0  792.48
#Mann=4,-1,0
  4462.6    0.16       0  4690.0     0.1       0  4990.2    0.07       0
  4996.2     0.1       0
Bank Sta=4990.2,4996.2
Exp/Cntr=0.3,0.1

Type RM Length L Ch R = 1,12384,287,287,287
BEGIN DESCRIPTION:
UNT 043 in HW 28.0
END DESCRIPTION:
XS GIS Cut Line= 3
      1983825.00     13631175.00      1983475.00     13631175.00
      1982832.68     13631235.93
#Sta/Elev= 30
  4665.8  792.33  4715.8  790.86  4755.8  788.58  4765.8  788.77  4835.8  781.05
  4945.8  775.86  4985.8  775.84  4992.8  770.83  4993.3  770.03  4998.3  770.03
  4998.8  770.83  5005.8  771.03  5013.3  774.32  5018.3  774.32  5025.8  775.40
  5064.9  777.25  5069.9  776.92  5126.3  779.13  5166.5  781.75  5178.1  781.05
  5246.8  781.70  5327.2  783.56  5367.4  785.32  5377.4  785.45  5397.5  784.49
  5417.6  784.63  5558.2  787.32  5595.8  789.06  5638.6  788.34  5661.0  788.94
#Mann=3,-1,0
  4665.8     0.1       0  4992.8    0.07       0  4998.8     0.1       0
Bank Sta=4992.8,4998.8
Exp/Cntr=0.3,0.1

Type RM Length L Ch R = 1,12097,273,273,273
BEGIN DESCRIPTION:
UNT 043 in HW 27.0
END DESCRIPTION:
XS GIS Cut Line= 3
      1983994.23     13631097.92      1983575.00     13630925.00
      1982811.87     13630952.07
#Sta/Elev= 30
  4532.3  789.32  4695.0  783.97  4710.2  784.15  4715.6  783.59  4747.8  783.48
  4787.4  782.54  4816.7  781.11  4834.3  780.85  4856.0  779.34  4877.6  776.73
  4947.2  774.79  4953.3  773.92  4964.2  773.54  4988.3  773.81  4992.8  769.72
  4993.3  768.92  4998.3  768.92  4998.8  769.72  5005.8  773.95  5025.8  773.70
  5080.3  775.01  5155.9  777.27  5215.9  778.35  5266.0  780.50  5366.0  780.83
  5476.1  783.42  5606.2  784.53  5676.2  786.24  5726.3  785.93  5749.4  786.35
#Mann=5,-1,0
  4532.3     0.1       0  4695.0    0.16       0  4992.8    0.07       0
  4998.8    0.16       0  5080.3     0.1       0
Bank Sta=4992.8,4998.8
Exp/Cntr=0.3,0.1

Type RM Length L Ch R = 1,11824,258,258,258
BEGIN DESCRIPTION:
UNT 043 in HW 26.0
END DESCRIPTION:
XS GIS Cut Line= 3
      1984025.00     13630925.00      1983625.00     13630675.00
      1982799.48     13630577.14
#Sta/Elev= 30
  4514.0  791.09  4564.1  790.06  4579.4  787.78  4585.3  787.91  4616.0  785.26
  4658.5  783.42  4673.8  781.83  4695.0  780.89  4710.3  779.16  4752.8  776.50
  4904.9  772.92  4972.1  773.08  4978.0  772.63  4979.8  769.32  4980.3  768.52
  4985.3  768.52  4985.8  769.32  4995.8  769.84  5005.8  773.16  5015.9  773.06
  5029.6  770.78  5038.1  771.33  5112.3  774.41  5217.6  777.33  5277.7  778.24
  5318.0  779.94  5338.1  779.62  5378.4  780.57  5569.8  780.85  5817.0  783.32
#Mann=5,-1,0
  4514.0     0.1       0  4979.8    0.07       0  4985.8     0.1       0
  5038.1    0.16       0  5217.6     0.1       0
Bank Sta=4979.8,4985.8
Exp/Cntr=0.3,0.1

Type RM Length L Ch R = 1,11566,320,320,320
BEGIN DESCRIPTION:
UNT 043 in HW 25.0
END DESCRIPTION:
XS GIS Cut Line= 3
      1984025.02     13630875.02      1983725.00     13630475.00
      1983225.02     13630175.01
#Sta/Elev= 30
  4460.2  791.38  4488.4  790.19  4496.7  790.42  4502.9  789.37  4522.2  788.31
  4563.2  785.85  4596.7  783.37  4682.1  774.69  4702.9  773.57  4796.7  771.79
  4896.7  770.88  4983.6  771.66  4992.2  766.22  4992.7  765.42  4997.7  765.42
  4998.2  766.22  5004.9  768.70  5008.9  769.49  5026.3  770.46  5032.1  771.80
  5041.9  770.71  5053.5  772.36  5076.8  771.80  5090.5  773.28  5127.3  773.89
  5275.1  774.69  5323.7  775.81  5403.4  779.01  5478.2  783.86  5543.3  787.91
#Mann=8,-1,0
  4460.2     0.1       0  4522.2    0.16       0  4563.2     0.1       0
  4992.2    0.07       0  4998.2     0.1       0  5008.9    0.16       0
  5127.3     0.1       0  5478.2    0.16       0
Bank Sta=4992.2,4998.2
Exp/Cntr=0.3,0.1

Type RM Length L Ch R = 1,11246,275,275,275
BEGIN DESCRIPTION:
UNT 043 in HW 24.0
END DESCRIPTION:
XS GIS Cut Line= 3
      1984327.53     13630827.09      1983975.00     13630375.00
      1983359.37     13630077.36
#Sta/Elev= 30
  4438.8  784.89  4484.7  783.72  4499.2  782.82  4561.8  781.44  4616.9  779.82
  4712.7  777.05  4727.1  775.91  4733.5  776.05  4770.6  774.23  4776.9  774.42
  4791.4  772.86  4841.1  770.89  4934.3  768.64  4975.9  769.41  4984.0  768.98
  4990.4  767.45  4995.5  763.69  4996.0  762.89  5001.0  762.89  5001.5  763.69
  5004.9  765.03  5008.9  769.85  5071.4  769.49  5226.5  771.40  5445.3  772.47
  5506.2  773.37  5589.7  776.32  5611.9  777.69  5657.2  782.26  5695.9  784.89
#Mann=7,-1,0
  4438.8     0.1       0  4561.8    0.16       0  4616.9     0.1       0
  4995.5    0.07       0  5001.5     0.1       0  5226.5    0.16       0
  5657.2     0.1       0
Bank Sta=4995.5,5001.5
Exp/Cntr=0.3,0.1

Type RM Length L Ch R = 1,10971,197,197,197
BEGIN DESCRIPTION:
UNT 043 in HW 23.0
END DESCRIPTION:
XS GIS Cut Line= 3
      1984856.14     13630741.11      1984175.00     13630225.00
      1983413.46     13629962.49
#Sta/Elev= 30
  4163.5  782.56  4276.4  782.33  4282.7  781.20  4297.2  781.42  4318.1  779.94
  4411.6  780.25  4623.0  776.83  4646.7  775.42  4675.8  775.97  4717.5  774.48
  4725.8  775.33  4786.8  773.89  4910.9  770.04  4967.9  766.81  4975.4  767.70
  4981.7  766.34  4993.3  761.41  4993.8  760.61  4998.8  760.61  4999.3  761.41
  5010.8  768.31  5014.9  767.43  5028.4  768.52  5071.0  767.53  5427.5  770.54
  5558.9  771.05  5631.6  772.74  5747.9  777.51  5798.0  782.20  5823.6  783.54
#Mann=6,-1,0
  4163.5     0.1       0  4623.0    0.05       0  4786.8     0.1       0
  4993.3    0.07       0  4999.3     0.1       0  5427.5    0.16       0
Bank Sta=4993.3,4999.3
Exp/Cntr=0.3,0.1

Type RM Length L Ch R = 1,10774,315,315,315
BEGIN DESCRIPTION:
UNT 043 in HW 22.0
END DESCRIPTION:
XS GIS Cut Line= 3
      1984918.68     13630436.45      1984416.06     13630116.13
      1983430.78     13629819.77
#Sta/Elev= 30
  4252.3  777.90  4387.1  775.91  4466.6  775.87  4545.3  773.82  4654.5  773.41
  4748.4  770.52  4761.5  771.84  4790.7  770.64  4800.1  771.64  4827.1  772.20
  4842.4  771.30  4846.0  769.27  4872.7  769.22  4905.6  769.05  4964.3  766.60
  4976.8  766.93  4985.2  762.98  4992.6  762.16  4993.1  761.36  4998.1  761.36
  4998.6  762.16  5004.6  766.43  5009.9  766.75  5075.9  766.34  5180.2  767.61
  5531.3  769.52  5590.8  770.76  5682.3  774.28  5767.7  777.84  5877.2  785.87
#Mann=6,-1,0
  4252.3     0.1       0  4761.5    0.05       0  4872.7     0.1       0
  4992.6    0.07       0  4998.6     0.1       0  5682.3    0.16       0
Bank Sta=4992.6,4998.6
Exp/Cntr=0.3,0.1

Type RM Length L Ch R = 1,10459,297,297,297
BEGIN DESCRIPTION:
UNT 043 in HW 21.0
END DESCRIPTION:
XS GIS Cut Line= 3
      1985046.28     13630207.29      1984425.00     13629825.00
      1983609.37     13629540.82
#Sta/Elev= 30
  4243.3  775.96  4336.8  775.03  4485.9  773.40  4494.7  773.12  4681.1  769.63
  4726.2  769.99  4835.6  767.56  4864.5  767.43  4878.8  766.10  4885.8  767.64
  4914.1  768.88  4937.6  765.68  4967.6  764.17  4983.0  763.48  4991.0  759.50
  4991.5  758.70  4996.5  758.70  4997.0  759.50  5004.5  762.81  5014.1  764.84
  5025.7  763.86  5045.2  764.83  5050.5  764.31  5288.5  764.96  5324.9  765.75
  5443.9  766.21  5506.1  767.60  5744.2  776.92  5830.5  783.45  5836.5  784.48
#Mann=8,-1,0
  4243.3    0.05       0  4336.8     0.1       0  4485.9    0.05       0
  4494.7     0.1       0  4835.6    0.05       0  4967.6     0.1       0
  4991.0    0.07       0  4997.0     0.1       0
Bank Sta=4991,4997
Exp/Cntr=0.3,0.1

Type RM Length L Ch R = 1,10162,225,225,225
BEGIN DESCRIPTION:
UNT 043 in HW 20.0
END DESCRIPTION:
XS GIS Cut Line= 3
      1985227.68     13629981.14      1984525.00     13629575.00
      1983624.96     13629374.99
#Sta/Elev= 30
  4163.6  772.12  4281.1  771.26  4308.4  770.54  4319.2  770.91  4404.6  770.71
  4726.1  766.12  4857.5  765.59  4871.3  765.75  4886.9  763.59  4902.7  764.67
  4924.2  764.93  4940.0  763.06  4977.8  762.83  4983.6  761.60  4996.5  758.02
  4997.0  757.22  5002.0  757.22  5002.5  758.02  5005.9  761.08  5016.2  762.11
  5091.7  761.45  5178.8  762.00  5276.1  761.64  5477.2  764.11  5552.7  767.30
  5579.6  770.17  5702.5  779.72  5780.6  783.80  5785.8  784.52  5897.2  789.77
#Mann=6,-1,0
  4163.6    0.05       0  4319.2     0.1       0  4857.5    0.05       0
  4983.6     0.1       0  4996.5    0.07       0  5002.5     0.1       0
Bank Sta=4996.5,5002.5
Exp/Cntr=0.3,0.1

Type RM Length L Ch R = 1,9937,350,350,350
BEGIN DESCRIPTION:
UNT 043 in HW 19.0
END DESCRIPTION:
XS GIS Cut Line= 3
      1985425.03     13629074.99      1984425.00     13629375.00
      1983724.97     13629275.00
#Sta/Elev= 30
  3969.0  779.90  4023.8  779.79  4167.4  774.57  4260.5  772.14  4522.4  760.85
  4612.0  759.32  4682.8  759.35  4699.8  758.80  4710.3  760.45  4721.6  760.46
  4741.6  759.56  4749.4  758.18  4772.9  759.34  4826.8  759.89  4898.2  760.53
  4950.4  759.99  4981.7  761.08  4991.3  759.13  4993.5  757.74  4994.0  756.94
  4999.0  756.94  4999.5  757.74  5002.6  760.31  5010.4  760.82  5194.9  759.39
  5275.7  760.50  5396.9  764.24  5447.4  766.83  5568.6  777.02  5720.2  786.98
#Mann=5,-1,0
  3969.0     0.1       0  4682.8    0.05       0  4826.8     0.1       0
  4993.5    0.07       0  4999.5     0.1       0
Bank Sta=4993.5,4999.5
Exp/Cntr=0.3,0.1

Type RM Length L Ch R = 1,9587,343,343,343
BEGIN DESCRIPTION:
UNT 043 in HW 18.0
END DESCRIPTION:
XS GIS Cut Line= 3
      1985325.03     13628975.00      1984541.93     13629095.73
      1983734.67     13629078.37
#Sta/Elev= 30
  3949.3  778.72  4051.7  776.77  4222.5  768.08  4246.2  766.20  4263.0  762.60
  4273.1  761.56  4309.4  759.22  4394.5  756.84  4485.8  756.30  4526.1  756.11
  4536.2  757.79  4566.5  756.31  4574.2  755.15  4574.7  754.35  4579.8  754.35
  4580.3  755.15  4586.8  756.22  4614.1  756.26  4758.6  758.41  4888.6  757.68
  4988.6  759.22  4998.6  756.87  5010.9  758.96  5018.6  758.17  5038.6  758.36
  5078.7  760.61  5118.7  761.64  5298.7  770.42  5448.7  778.81  5549.1  780.85
#Mann=5,-1,0
  3949.3     0.1       0  4485.8    0.05       0  4574.2    0.07       0
  4580.3    0.05       0  4614.1     0.1       0
Bank Sta=4574.2,4580.3
Exp/Cntr=0.3,0.1

Type RM Length L Ch R = 1,9244,291,291,291
BEGIN DESCRIPTION:
UNT 043 in HW 17.0
END DESCRIPTION:
XS GIS Cut Line= 3
      1985354.10     13628866.33      1984668.33     13628829.44
      1984082.35     13628792.55
#Sta/Elev= 30
  4104.3  776.86  4173.5  777.14  4220.4  775.95  4225.4  776.34  4263.6  773.60
  4393.8  768.17  4408.6  768.11  4453.9  765.40  4544.0  758.71  4614.7  755.14
  4684.2  755.15  4694.3  754.13  4714.3  755.36  4734.3  755.47  4744.3  755.12
  4751.3  753.90  4751.8  753.10  4756.9  753.10  4757.4  753.90  4767.4  754.97
  4874.6  756.19  4934.7  756.17  4984.8  757.37  4994.8  754.80  5004.8  754.70
  5014.8  757.76  5054.9  756.62  5085.0  756.72  5165.1  760.23  5378.2  766.95
#Mann=5,-1,0
  4104.3     0.1       0  4614.7    0.05       0  4751.3    0.07       0
  4757.4    0.05       0  4767.4     0.1       0
Bank Sta=4751.3,4757.4
Exp/Cntr=0.3,0.1

Type RM Length L Ch R = 1,8953,97,97,97
BEGIN DESCRIPTION:
Mapping XS a381d310
END DESCRIPTION:
XS GIS Cut Line= 4
      1985345.37     13628844.62      1984684.25     13628714.08
      1984672.67     13628430.14      1984049.92     13628725.24
#Sta/Elev= 30
  4269.8  776.61  4331.3  776.76  4397.3  774.77  4596.4  766.03  4653.7  761.75
  4714.8  758.91  4779.8  754.11  4841.0  754.71  4864.0  753.68  4892.0  754.60
  4924.5  753.21  4932.7  754.42  4972.8  754.88  4999.8  750.58  5000.3  749.78
  5005.4  749.78  5005.9  750.58  5022.8  753.58  5042.8  754.42  5072.9  753.33
  5082.9  754.10  5227.9  753.28  5358.1  754.65  5365.6  754.12  5371.2  751.67
  5380.2  754.39  5388.4  755.21  5695.1  758.32  5800.7  765.63  5917.0  767.62
#Mann=5,-1,0
  4269.8     0.1       0  4714.8    0.05       0  4924.5     0.1       0
  4999.8    0.07       0  5005.9     0.1       0
Bank Sta=4999.8,5005.9
Exp/Cntr=0.3,0.1

Type RM Length L Ch R = 1,8856,674,674,674
BEGIN DESCRIPTION:
Mapping XS fe096b88
END DESCRIPTION:
XS GIS Cut Line= 4
      1985334.52     13628827.26      1984771.06     13628668.51
      1984763.82     13628334.65      1984073.15     13628650.75
#Sta/Elev= 30
  4363.1  776.41  4414.5  776.82  4445.7  776.01  4574.9  770.94  4657.4  766.85
  4794.6  758.85  4840.5  753.74  4923.6  754.40  4941.1  752.96  4982.0  753.58
  4989.0  749.38  4989.5  748.58  4994.6  748.58  4995.1  749.38  4997.2  749.45
  5002.2  752.34  5012.0  753.10  5103.3  752.43  5279.8  749.43  5291.0  750.44
  5319.5  751.03  5348.0  750.02  5354.6  751.71  5358.1  752.60  5402.1  753.63
  5532.1  754.18  5796.2  757.03  5876.2  759.85  5939.8  764.34  6042.0  767.35
#Mann=6,-1,0
  4363.1     0.1       0  4657.4    0.05       0  4989.0    0.04       0
  4995.1    0.05       0  5103.3    0.08       0  5354.6     0.1       0
Bank Sta=4989,4995.1
Exp/Cntr=0.3,0.1

Type RM Length L Ch R = 1,8182,485,485,485
BEGIN DESCRIPTION:
Mapping XS 6517e613
END DESCRIPTION:
XS GIS Cut Line= 3
      1985208.69     13628230.48      1984739.95     13628171.89
      1984054.17     13628629.80
#Sta/Elev= 30
  4656.6  775.31  4700.6  774.13  4738.5  771.16  4743.5  771.53  4824.2  764.33
  4861.9  759.30  4899.8  749.61  4922.3  747.81  4972.7  747.12  4985.4  745.77
  4989.8  742.37  4990.3  741.57  4995.4  741.57  4995.9  742.37  5003.0  742.98
  5013.0  745.92  5023.1  746.53  5061.0  747.41  5103.7  747.17  5113.8  748.52
  5136.4  748.76  5171.0  747.58  5184.3  748.95  5207.1  749.19  5244.2  750.25
  5689.0  756.65  5761.0  759.12  5833.1  763.60  5905.2  766.03  5953.6  766.40
#Mann=6,-1,0
  4656.6     0.1       0  4989.8    0.07       0  4995.9     0.1       0
  5136.4    0.05       0  5207.1    0.08       0  5244.2     0.1       0
Bank Sta=4989.8,4995.9
Exp/Cntr=0.3,0.1

Type RM Length L Ch R = 1,7697,320,320,320
BEGIN DESCRIPTION:
UNT 043 in HW 16.0
END DESCRIPTION:
XS GIS Cut Line= 3
      1985310.70     13627972.24      1984775.00     13627725.00
      1984132.29     13627668.41
#Sta/Elev= 30
  4427.4  771.03  4476.3  769.50  4504.8  766.58  4527.7  767.23  4533.3  765.97
  4573.6  764.30  4602.1  761.52  4619.5  761.05  4625.0  759.58  4648.0  757.68
  4775.1  749.27  4911.4  745.33  4928.8  743.86  4973.3  743.51  4980.2  741.71
  4985.7  741.69  4992.0  738.83  4992.5  738.03  4998.8  738.83  5003.2  741.77
  5008.7  741.70  5014.6  744.40  5027.4  743.84  5044.5  744.96  5107.7  743.49
  5143.0  744.26  5248.3  749.09  5569.5  753.14  5599.6  755.98  5662.6  758.17
#Mann=5,-1,0
  4427.4     0.1       0  4992.0    0.07       0  4998.8     0.1       0
  5044.5    0.05       0  5143.0     0.1       0
Bank Sta=4992,4998.8
Exp/Cntr=0.3,0.1

Type RM Length L Ch R = 1,7377,235,235,235
BEGIN DESCRIPTION:
UNT 043 in HW 15.0
END DESCRIPTION:
XS GIS Cut Line= 3
      1985443.08     13627776.93      1984852.79     13627436.21
      1984331.95     13627334.21
#Sta/Elev= 30
  4375.1  761.08  4389.6  761.02  4405.4  761.86  4411.1  760.95  4464.2  759.59
  4572.0  754.07  4580.7  753.91  4587.7  754.59  4593.5  753.37  4615.4  751.46
  4696.2  748.40  4791.7  743.34  4872.1  741.08  4984.1  741.06  4989.8  737.23
  5002.2  736.71  5002.7  735.91  5008.5  735.91  5009.0  736.71  5011.4  739.91
  5027.2  741.00  5153.7  743.24  5186.9  743.38  5197.6  742.49  5217.5  743.51
  5253.3  744.15  5380.5  746.33  5501.5  752.20  5558.1  752.91  5587.4  753.94
#Mann=5,-1,0
  4375.1     0.1       0  5002.2    0.07       0  5009.0     0.1       0
  5153.7    0.05       0  5253.3     0.1       0
Bank Sta=5002.2,5009
Exp/Cntr=0.3,0.1

Type RM Length L Ch R = 1,7142,474,474,474
BEGIN DESCRIPTION:
Mapping XS 921622bb
END DESCRIPTION:
XS GIS Cut Line= 3
      1985421.33     13627486.11      1984841.94     13627273.45
      1984339.20     13627182.44
#Sta/Elev= 30
  4626.6  753.46  4718.6  752.26  4788.6  749.21  4905.3  746.46  4930.4  745.92
  4935.7  746.64  4966.2  744.02  4974.2  739.31  4984.9  736.08  4988.0  733.90
  4988.5  733.10  4994.4  733.10  4994.9  733.90  5006.2  739.70  5052.4  739.41
  5123.4  741.23  5199.5  740.97  5324.4  742.22  5362.6  743.00  5371.6  741.15
  5376.7  741.09  5393.1  743.27  5423.9  743.17  5454.1  743.89  5488.7  747.05
  5494.7  748.32  5542.2  750.89  5555.7  749.93  5626.9  751.71  5754.7  753.13
#Mann=5,-1,0
  4626.6     0.1       0  4988.0    0.07       0  4994.9     0.1       0
  5324.4    0.05       0  5423.9     0.1       0
Bank Sta=4988,4994.9
Exp/Cntr=0.3,0.1

Type RM Length L Ch R = 1,6668,139,139,139
BEGIN DESCRIPTION:
UNT 043 in HW 14.0
END DESCRIPTION:
XS GIS Cut Line= 3
      1985374.98     13627374.96      1985154.44     13627017.38
      1984766.00     13626885.00
#Sta/Elev= 30
  4343.6  751.52  4357.1  750.58  4461.0  749.04  4503.8  747.75  4519.2  748.59
  4525.1  747.57  4561.8  746.47  4782.8  742.24  4863.0  739.87  4976.2  735.95
  4992.1  732.34  4992.6  731.54  4998.6  731.54  4999.1  732.34  5002.2  734.68
  5007.5  734.00  5016.7  735.73  5027.3  736.14  5033.6  735.43  5039.0  735.60
  5048.4  734.01  5064.9  738.76  5090.6  742.29  5096.3  743.87  5101.5  743.82
  5122.3  746.22  5127.6  746.09  5159.0  749.07  5165.4  750.24  5174.1  750.94
#Mann=6,-1,0
  4343.6     0.1       0  4863.0    0.16       0  4992.1    0.07       0
  4999.1    0.16       0  5039.0     0.1       0  5165.4    0.05       0
Bank Sta=4992.1,4999.1
Exp/Cntr=0.3,0.1

Type RM Length L Ch R = 1,6529,93,93,93
BEGIN DESCRIPTION:
UNT 043 in HW 13.0
END DESCRIPTION:
XS GIS Cut Line= 3
      1985501.64     13627123.70      1984975.00     13626825.00
      1984775.01     13626775.00
#Sta/Elev= 30
  4369.6  748.86  4417.6  748.35  4492.2  746.67  4526.7  744.72  4595.0  743.80
  4644.0  741.82  4719.0  741.18  4762.3  740.17  4771.7  740.47  4886.3  738.06
  4902.2  738.27  4917.6  737.68  4923.8  738.02  4929.6  737.38  4977.6  735.36
  4985.4  733.55  4989.6  730.23  4990.1  729.43  4996.1  729.43  4996.6  730.23
  4998.2  731.74  5006.0  733.80  5018.0  734.45  5026.6  735.27  5034.3  737.16
  5047.2  738.88  5109.1  743.94  5150.3  750.47  5178.4  753.75  5181.2  753.77
#Mann=6,-1,0
  4369.6     0.1       0  4771.7    0.16       0  4989.6    0.07       0
  4996.6    0.16       0  5018.0     0.1       0  5178.4    0.05       0
Bank Sta=4989.6,4996.6
Exp/Cntr=0.3,0.1

Type RM Length L Ch R = 1,6436,617,617,617
BEGIN DESCRIPTION:
Mapping XS 644b69ba
END DESCRIPTION:
XS GIS Cut Line= 3
      1985638.42     13626956.62      1984941.77     13626728.75
      1984779.47     13626720.09
#Sta/Elev= 30
  4342.2  747.39  4377.4  747.03  4545.7  742.07  4608.8  738.40  4622.7  736.84
  4648.5  737.08  4654.6  736.18  4681.2  736.90  4686.5  736.15  4713.1  737.22
  4718.3  736.41  4744.9  736.68  4750.2  736.02  4941.4  736.52  4978.5  734.57
  4987.6  732.98  4994.6  729.50  4995.1  728.70  5001.1  728.70  5001.6  729.50
  5010.4  734.00  5029.7  734.72  5042.2  738.12  5051.9  739.55  5082.0  742.22
  5142.0  744.42  5162.1  746.78  5192.1  751.87  5232.2  754.74  5237.7  755.80
#Mann=6,-1,0
  4342.2     0.1       0  4648.5    0.16       0  4994.6    0.07       0
  5001.6    0.16       0  5051.9     0.1       0  5237.7    0.08       0
Bank Sta=4994.6,5001.6
Exp/Cntr=0.3,0.1

Type RM Length L Ch R = 1,5819,47,47,47
BEGIN DESCRIPTION:
Mapping XS 652e3915
END DESCRIPTION:
XS GIS Cut Line= 4
      1985827.21     13626780.84      1985618.85     13626667.98
      1984811.56     13626687.51      1984765.98     13626624.57
#Sta/Elev= 30
  4679.5  748.02  4887.9  745.49  4913.7  745.85  4930.3  745.13  4950.3  741.94
  4970.3  736.42  4986.8  726.69  4987.3  725.89  4993.3  725.89  4993.8  726.69
  4997.6  729.56  5002.6  728.55  5010.3  730.97  5100.4  735.42  5200.4  737.36
  5310.4  741.27  5360.4  740.20  5386.6  741.02  5409.4  740.76  5414.4  736.50
  5420.5  738.25  5430.5  738.57  5460.5  736.23  5520.5  737.60  5590.5  742.23
  5650.5  745.14  5719.8  753.94  5774.7  758.46  5780.2  759.54  5801.7  760.68
#Mann=6,-1,0
  4679.5     0.1       0  4887.9    0.16       0  4986.8    0.07       0
  4993.8    0.16       0  5386.6     0.1       0  5774.7    0.08       0
Bank Sta=4986.8,4993.8
Exp/Cntr=0.3,0.1

Type RM Length L Ch R = 1,5772,65,65,65
BEGIN DESCRIPTION:
Mapping XS 89499871
END DESCRIPTION:
XS GIS Cut Line= 4
      1985868.40     13626722.23      1985638.38     13626628.92
      1984850.62     13626648.45      1984765.98     13626585.51
#Sta/Elev= 30
  4667.7  748.01  4777.0  746.55  4893.4  745.92  4929.3  744.07  4956.9  735.55
  4961.9  737.80  4969.3  734.70  4989.3  728.61  4995.8  728.18  4996.3  727.38
  5002.3  727.38  5002.8  728.18  5009.3  730.61  5099.4  735.81  5269.6  739.58
  5389.5  742.08  5449.5  741.94  5479.5  741.14  5509.5  741.52  5539.5  740.67
  5569.5  741.25  5659.5  745.24  5689.5  749.61  5703.9  750.64  5717.6  752.99
  5767.7  758.13  5773.9  758.25  5782.3  759.68  5787.8  759.79  5809.4  761.71
#Mann=6,-1,0
  4667.7     0.1       0  4893.4    0.16       0  4995.8    0.07       0
  5002.8    0.16       0  5269.6     0.1       0  5787.8    0.08       0
Bank Sta=4995.8,5002.8
Exp/Cntr=0.3,0.1

Type RM Length L Ch R = 1,5707,292,292,292
BEGIN DESCRIPTION:
UNT 043 in HW 12.0
END DESCRIPTION:
XS GIS Cut Line= 3
      1985902.72     13626707.78      1985575.00     13626575.00
      1984831.33     13626369.65
#Sta/Elev= 30
  4650.5  748.04  4721.3  747.70  4780.3  746.45  4903.9  745.86  4928.6  744.54
  4935.7  742.60  4941.1  739.77  4959.8  734.03  4965.2  731.81  4982.5  729.34
  4985.8  728.25  4986.3  727.45  4992.3  727.45  4992.8  728.25  5006.7  729.30
  5014.5  730.76  5021.3  731.19  5026.5  730.74  5045.6  731.90  5065.1  733.95
  5076.7  735.11  5118.2  736.74  5327.2  740.26  5356.3  741.24  5481.3  742.68
  5616.2  746.77  5647.3  748.32  5688.8  752.23  5736.1  760.41  5775.6  764.09
#Mann=5,-1,0
  4650.5     0.1       0  4903.9    0.16       0  4985.8    0.07       0
  4992.8    0.16       0  5065.1     0.1       0
Bank Sta=4985.8,4992.8
Exp/Cntr=0.3,0.1

Type RM Length L Ch R = 1,5415,327,327,327
BEGIN DESCRIPTION:
Mapping XS e3a75214
END DESCRIPTION:
XS GIS Cut Line= 3
      1986048.55     13626567.16      1985931.35     13626390.06
      1984953.32     13626189.77
#Sta/Elev= 30
  4429.8  746.82  4528.3  746.21  4642.2  743.89  4679.3  744.32  4794.3  742.20
  4832.4  742.55  4903.8  740.48  4924.3  738.79  4944.6  735.67  4985.5  727.11
  4987.5  724.23  4988.0  723.43  4994.0  723.43  4994.5  724.23  5005.9  727.08
  5016.1  728.37  5026.3  729.32  5047.2  729.33  5137.2  734.24  5142.3  733.70
  5288.5  738.74  5394.5  740.30  5485.2  742.79  5506.1  744.21  5516.3  745.97
  5535.6  745.14  5540.7  745.97  5591.2  747.11  5636.5  750.08  5640.5  749.70
#Mann=5,-1,0
  4429.8     0.1       0  4944.6    0.16       0  4987.5    0.07       0
  4994.5    0.16       0  5047.2     0.1       0
Bank Sta=4987.5,4994.5
Exp/Cntr=0.3,0.1

Type RM Length L Ch R = 1,5088,213,213,213
BEGIN DESCRIPTION:
UNT 043 in HW 11.0
END DESCRIPTION:
XS GIS Cut Line= 3
      1986092.81     13626288.49      1985913.12     13626080.16
      1985148.72     13625939.76
#Sta/Elev= 30
  4434.6  741.16  4492.0  741.50  4584.5  740.84  4605.8  740.22  4758.6  738.82
  4779.0  737.77  4799.3  737.59  4840.0  735.30  4860.3  735.12  4890.8  732.94
  4901.0  732.01  4929.2  727.55  4951.8  726.85  4972.2  727.64  4982.3  726.65
  4989.0  722.70  4989.5  721.90  4995.5  721.90  4996.0  722.70  5002.7  725.31
  5012.8  728.14  5023.0  728.62  5098.7  729.76  5185.7  733.43  5263.0  736.13
  5277.2  736.14  5368.7  738.78  5389.0  738.93  5409.3  739.95  5486.9  742.07
#Mann=3,-1,0
  4434.6     0.1       0  4989.0    0.07       0  4996.0     0.1       0
Bank Sta=4989,4996
Exp/Cntr=0.3,0.1

Type RM Length L Ch R = 1,4875,74,74,74
BEGIN DESCRIPTION:
UNT 043 in HW 10.0
END DESCRIPTION:
XS GIS Cut Line= 3
      1986155.29     13625849.26      1985552.01     13625827.56
      1985228.20     13625745.53
#Sta/Elev= 30
  4515.2  735.56  4585.5  735.69  4685.6  734.92  4845.7  732.35  4915.7  729.42
  4935.8  728.06  4955.8  725.83  4985.8  726.22  4992.3  722.65  4992.8  721.85
  4998.8  721.85  4999.3  722.65  5015.8  726.01  5045.8  726.79  5055.9  727.67
  5075.8  727.49  5095.9  728.10  5136.4  730.46  5208.6  732.79  5227.6  733.21
  5232.8  732.30  5239.6  733.28  5268.6  734.63  5273.7  734.24  5309.6  736.00
  5314.7  735.73  5355.7  738.14  5373.7  738.20  5396.7  739.70  5452.9  741.21
#Mann=3,-1,0
  4515.2     0.1       0  4992.3    0.07       0  4999.3     0.1       0
Bank Sta=4992.3,4999.3
Exp/Cntr=0.3,0.1

Type RM Length L Ch R = 1,4801,233,233,233
BEGIN DESCRIPTION:
Mapping XS 2b626359
END DESCRIPTION:
XS GIS Cut Line= 3
      1986164.00     13625762.46      1985586.73     13625762.46
      1985265.52     13625640.92
#Sta/Elev= 30
  4516.8  734.97  4635.8  733.75  4685.8  733.89  4755.8  732.21  4805.8  732.22
  4845.8  731.38  4905.8  729.38  4965.8  725.84  4985.8  726.11  4992.3  721.50
  4992.8  720.70  4998.8  720.70  4999.3  721.50  5005.8  723.68  5015.8  725.51
  5025.8  726.08  5092.4  727.71  5101.1  727.46  5106.6  728.57  5156.1  730.25
  5161.5  729.53  5234.9  731.96  5246.6  733.06  5266.1  733.69  5296.3  737.18
  5301.6  737.06  5326.4  739.29  5386.8  741.60  5406.0  741.52  5437.5  743.31
#Mann=3,-1,0
  4516.8     0.1       0  4992.3    0.07       0  4999.3     0.1       0
Bank Sta=4992.3,4999.3
Exp/Cntr=0.3,0.1

Type RM Length L Ch R = 1,4568,318,318,318
BEGIN DESCRIPTION:
Mapping XS 22961083
END DESCRIPTION:
XS GIS Cut Line= 2
      1986198.69     13625714.71      1985321.96     13625432.59
#Sta/Elev= 30
  4477.0  733.88  4553.4  733.14  4660.2  730.93  4783.2  729.87  4922.1  725.72
  4943.1  725.26  4964.1  723.90  4981.0  723.88  4983.8  722.57  4986.2  721.44
  4992.1  719.98  4992.6  719.18  4998.6  719.18  4999.1  719.98  5006.1  722.45
  5013.0  724.05  5027.1  724.70  5058.7  728.30  5090.2  730.55  5109.3  731.24
  5132.2  733.09  5141.4  732.94  5146.6  733.75  5205.5  737.16  5242.9  740.82
  5274.9  743.01  5307.0  744.43  5312.3  745.27  5376.4  747.37  5398.0  747.57
#Mann=5,-1,0
  4477.0     0.1       0  4922.1    0.12       0  4983.8     0.1       0
  4992.1    0.07       0  4999.1     0.1       0
Bank Sta=4992.1,4999.1
Exp/Cntr=0.3,0.1

Type RM Length L Ch R = 1,4250,351,351,351
BEGIN DESCRIPTION:
Mapping XS 2e38dab7
END DESCRIPTION:
XS GIS Cut Line= 2
      1986272.53     13625627.93      1985613.58     13625129.38
#Sta/Elev= 30
  4582.3  732.20  4611.3  732.14  4717.4  729.69  4746.6  729.92  4767.4  728.25
  4922.7  725.23  4940.0  724.54  4961.9  722.28  4990.0  722.95  4992.7  719.82
  4993.3  719.02  4999.3  719.02  4999.8  719.82  5004.5  720.10  5010.8  721.75
  5025.6  723.41  5046.2  727.88  5054.5  730.21  5060.7  732.89  5081.6  737.39
  5110.7  739.94  5139.8  741.73  5160.6  742.55  5175.2  743.79  5210.6  744.48
  5225.1  745.39  5275.1  745.33  5318.7  746.30  5331.6  745.78  5408.6  746.12
#Mann=6,-1,0
  4582.3     0.1       0  4922.7    0.12       0  4961.9    0.07       0
  4992.7    0.07       0  4999.8    0.07       0  5025.6     0.1       0
Bank Sta=4992.7,4999.8
Exp/Cntr=0.3,0.1

Type RM Length L Ch R = 1,3899,253,253,253
BEGIN DESCRIPTION:
UNT 043 in HW 9.0
END DESCRIPTION:
XS GIS Cut Line= 3
      1986428.76     13625671.35      1986361.28     13625524.65
      1986017.12     13624748.40
#Sta/Elev= 30
  4499.3  732.54  4641.9  731.36  4763.5  727.58  4885.3  722.60  4890.8  723.01
  4955.1  721.54  4977.6  721.82  4983.9  721.51  4995.9  719.58  4996.5  718.78
  5002.5  718.78  5003.0  719.58  5007.2  720.76  5030.4  721.93  5048.6  724.03
  5067.5  725.46  5111.2  726.56  5129.0  726.04  5163.6  727.26  5174.5  727.24
  5181.0  726.38  5186.5  727.34  5204.3  727.26  5256.3  728.84  5279.6  728.94
  5302.9  729.62  5308.3  730.21  5378.2  731.29  5430.2  733.23  5509.9  735.33
#Mann=5,-1,0
  4499.3     0.1       0  4995.9    0.07       0  5003.0     0.1       0
  5048.6    0.07       0  5067.5     0.1       0
Bank Sta=4995.9,5003
Exp/Cntr=0.3,0.1

Type RM Length L Ch R = 1,3646,407,407,407
BEGIN DESCRIPTION:
UNT 043 in HW 8.0
END DESCRIPTION:
XS GIS Cut Line= 3
      1986480.83     13625640.91      1986461.63     13625264.06
      1986394.04     13624629.79
#Sta/Elev= 30
  4562.8  731.83  4638.8  731.62  4668.8  731.01  4678.9  730.23  4688.9  730.65
  4718.9  730.09  4809.0  727.96  4888.2  725.04  4899.1  723.94  4919.2  723.00
  4937.2  720.76  4954.9  719.72  4979.4  720.31  4989.5  719.82  4996.0  716.99
  4996.5  716.19  5002.6  716.19  5003.1  716.99  5009.6  719.85  5019.6  720.49
  5039.8  720.22  5059.9  722.10  5086.7  723.80  5170.5  726.34  5251.0  727.53
  5452.1  729.29  5512.4  730.22  5519.6  730.95  5532.5  730.62  5578.0  731.98
#Mann=5,-1,0
  4562.8     0.1       0  4888.2    0.12       0  4996.0    0.07       0
  5003.1    0.12       0  5086.7     0.1       0
Bank Sta=4996,5003.1
Exp/Cntr=0.3,0.1

Type RM Length L Ch R = 1,3239,391,391,391
BEGIN DESCRIPTION:
UNT 043 in HW 7.0
END DESCRIPTION:
XS GIS Cut Line= 3
      1986511.20     13625662.65      1986836.73     13625167.84
      1986715.21     13624642.70
#Sta/Elev= 30
  4350.0  731.05  4516.2  730.43  4582.5  727.78  4588.5  728.42  4597.6  727.65
  4603.5  728.05  4639.7  726.26  4754.8  724.45  4865.0  722.20  4870.8  721.97
  4892.7  720.89  4913.8  720.79  4928.9  719.36  4934.9  719.59  4965.7  717.79
  4980.7  718.34  4986.3  718.75  4993.0  714.87  4993.5  714.07  4999.6  714.07
  5000.1  714.87  5006.8  718.38  5022.2  718.13  5056.9  718.46  5104.8  721.52
  5201.8  724.77  5345.5  727.58  5396.8  727.59  5414.0  728.54  5481.3  729.94
#Mann=8,-1,0
  4350.0     0.1       0  4754.8    0.07       0  4865.0     0.1       0
  4870.8    0.12       0  4980.7    0.16       0  4993.0    0.07       0
  5000.1    0.16       0  5022.2     0.1       0
Bank Sta=4993,5000.1
Exp/Cntr=0.3,0.1

Type RM Length L Ch R = 1,2848,421,421,421
BEGIN DESCRIPTION:
UNT 043 in HW 6.0
END DESCRIPTION:
XS GIS Cut Line= 3
      1987375.01     13625575.03      1987153.57     13624955.16
      1987027.72     13624603.64
#Sta/Elev= 30
  4394.2  734.96  4440.4  734.23  4465.9  729.43  4471.2  729.62  4496.7  723.14
  4527.5  721.13  4614.5  716.89  4638.5  718.40  4686.0  718.85  4700.8  718.92
  4855.6  721.41  4942.6  716.74  4978.7  717.31  4995.3  713.51  4995.9  712.71
  5002.0  712.71  5002.5  713.51  5004.2  715.31  5010.1  717.51  5039.5  716.84
  5137.6  721.16  5152.8  722.83  5158.8  727.16  5170.7  724.65  5178.2  722.89
  5190.7  722.64  5296.0  724.09  5301.3  724.97  5362.8  724.67  5425.8  725.91
#Mann=7,-1,0
  4394.2     0.1       0  4686.0    0.12       0  4700.8     0.1       0
  4995.3    0.07       0  5002.5     0.1       0  5039.5    0.16       0
  5170.7     0.1       0
Bank Sta=4995.3,5002.5
Exp/Cntr=0.3,0.1

Type RM Length L Ch R = 1,2427,296,296,296
BEGIN DESCRIPTION:
UNT 043 in HW 5.0
END DESCRIPTION:
XS GIS Cut Line= 3
      1987737.12     13625565.17      1987531.39     13624901.13
      1987140.76     13624593.83
#Sta/Elev= 30
  4379.0  735.84  4404.2  734.83  4431.5  732.61  4442.0  730.98  4474.6  728.01
  4494.3  726.91  4515.3  723.85  4588.6  719.57  4637.6  718.06  4766.5  717.41
  4876.3  715.99  4892.2  715.11  4953.6  713.96  4986.4  713.62  4992.9  711.33
  4993.5  710.53  5000.1  710.53  5000.7  711.33  5006.7  712.94  5011.9  712.31
  5017.8  714.21  5028.3  714.16  5049.8  715.91  5148.6  718.02  5254.0  719.15
  5311.3  720.66  5367.9  720.77  5425.7  722.40  5517.0  723.02  5571.2  724.54
#Mann=5,-1,0
  4379.0     0.1       0  4953.6    0.16       0  4992.9    0.07       0
  5000.7    0.16       0  5148.6     0.1       0
Bank Sta=4992.9,5000.7
Exp/Cntr=0.3,0.1

Type RM Length L Ch R = 1,2131,444,444,444
BEGIN DESCRIPTION:
UNT 043 in HW 4.0
END DESCRIPTION:
XS GIS Cut Line= 3
      1987997.57     13625067.82      1987752.75     13624833.42
      1987172.06     13624471.46
#Sta/Elev= 30
  4731.2  732.06  4798.7  731.34  4862.2  728.44  4883.6  726.36  4890.5  726.42
  4897.8  725.20  4904.7  725.51  4911.9  723.97  4918.8  723.75  4926.1  721.94
  4933.0  722.36  4940.2  720.12  4947.1  718.92  4961.3  714.66  4975.4  712.34
  4989.6  711.37  4999.8  709.66  5000.5  708.86  5007.1  708.86  5007.7  709.66
  5011.0  712.19  5020.8  712.36  5090.3  713.63  5096.2  714.18  5139.9  714.42
  5279.1  715.21  5400.6  716.59  5574.2  720.61  5662.6  722.10  5754.4  722.85
#Mann=5,-1,0
  4731.2     0.1       0  4999.8    0.07       0  5007.7     0.1       0
  5020.8    0.16       0  5139.9     0.1       0
Bank Sta=4999.8,5007.7
Exp/Cntr=0.3,0.1

Type RM Length L Ch R = 1,1687,214,214,214
BEGIN DESCRIPTION:
Mapping XS 4b66a389
END DESCRIPTION:
XS GIS Cut Line= 3
      1988086.11     13624614.68      1987916.81     13624552.17
      1987169.70     13624398.58
#Sta/Elev= 30
  4641.7  719.33  4706.8  718.84  4749.5  717.68  4773.4  717.44  4809.0  716.22
  4926.1  712.63  4931.7  711.93  4956.7  710.71  4982.1  710.10  4993.6  708.64
  4994.3  707.84  5000.9  707.84  5001.5  708.64  5027.3  710.57  5040.9  710.41
  5058.8  710.54  5077.7  711.39  5099.7  711.73  5128.0  713.23  5150.7  713.61
  5160.9  714.63  5183.5  715.37  5222.2  715.98  5233.9  715.75  5324.3  717.93
  5365.1  719.32  5430.2  719.95  5497.8  721.34  5530.9  721.51  5584.9  723.24
#Mann=5,-1,0
  4641.7     0.1       0  4809.0    0.16       0  4993.6    0.07       0
  5001.5    0.16       0  5040.9     0.1       0
Bank Sta=4993.6,5001.5
Exp/Cntr=0.3,0.1

Type RM Length L Ch R = 1,1473,267,267,267
BEGIN DESCRIPTION:
UNT 043 in HW 3.0
END DESCRIPTION:
XS GIS Cut Line= 3
      1988172.05     13624507.91      1987775.00     13624325.00
      1987382.99     13624211.03
#Sta/Elev= 30
  4538.1  719.76  4567.9  719.48  4611.9  719.73  4628.6  718.85  4645.0  718.36
  4667.0  718.32  4751.7  715.50  4854.1  711.68  4931.2  710.52  4977.9  708.52
  4985.7  706.53  4988.1  702.03  4988.7  701.23  4995.3  701.23  4996.0  702.03
  5006.5  708.04  5012.3  708.58  5030.8  711.00  5037.7  711.53  5089.8  713.30
  5103.0  713.09  5131.4  713.59  5175.3  713.30  5208.8  713.64  5242.4  714.88
  5247.6  714.62  5281.1  715.10  5348.2  716.84  5360.6  716.79  5383.5  717.62
#Mann=5,-1,0
  4538.1     0.1       0  4751.7    0.16       0  4988.1    0.07       0
  4996.0    0.16       0  5012.3     0.1       0
Bank Sta=4988.1,4996
Exp/Cntr=0.3,0.1

Type RM Length L Ch R = 1,1206,388,388,388
BEGIN DESCRIPTION:
Mapping XS 3e72288c
END DESCRIPTION:
XS GIS Cut Line= 2
      1988242.32     13624231.85      1987435.04     13623916.75
#Sta/Elev= 30
  4636.1  715.65  4639.9  716.04  4645.3  715.61  4664.4  715.73  4669.7  715.25
  4676.2  715.54  4748.6  714.47  4753.9  714.04  4772.8  714.42  4832.8  711.54
  4838.1  712.26  4862.6  711.88  4911.6  709.75  4917.0  709.99  4946.8  708.77
  4971.3  708.42  4976.7  704.72  4991.8  701.43  4992.5  700.63  4999.1  700.63
  4999.7  701.43  5008.9  707.00  5025.6  708.58  5080.0  710.17  5127.0  711.09
  5194.0  710.83  5288.0  712.32  5411.4  712.89  5416.9  713.41  5502.7  714.98
#Mann=3,-1,0
  4636.1     0.1       0  4991.8    0.07       0  4999.7     0.1       0
Bank Sta=4991.8,4999.7
Exp/Cntr=0.3,0.1

Type RM Length L Ch R = 1,818,86,86,86
BEGIN DESCRIPTION:
UNT 043 in HW 2.0
END DESCRIPTION:
XS GIS Cut Line= 3
      1988315.25     13624499.17      1988306.57     13623739.67
      1987473.22     13623752.69
#Sta/Elev= 30
  3971.2  718.93  4015.4  719.18  4095.4  718.42  4195.4  716.43  4325.4  712.44
  4385.4  711.33  4495.4  711.36  4535.4  710.57  4677.4  709.99  4725.4  709.78
  4754.6  710.74  4792.3  709.60  4862.3  709.64  4962.3  707.84  4972.3  707.16
  4982.3  702.34  4988.4  697.86  4989.1  697.06  4995.7  697.06  4996.4  697.86
  5002.4  701.64  5012.4  704.94  5022.4  706.51  5032.4  707.00  5162.4  709.63
  5182.4  709.48  5202.4  710.32  5321.3  711.78  5432.4  713.25  5564.2  715.75
#Mann=5,-1,0
  3971.2     0.1       0  4677.4    0.05       0  4988.4    0.04       0
  4996.4    0.05       0  5321.3     0.1       0
Bank Sta=4988.4,4996.4
Exp/Cntr=0.3,0.1
