--- UNT 006 in La Jarita Watershed.prj (project) ---

Proj Title=UNT 006 in La Jarita Watershed Base Level Engineering
Current Plan=p01
Default Exp/Contr=0.3,0.1
English Units
Geom File=g01
Flow File=f01
Plan File=p01
Y Axis Title=Elevation
X Axis Title(PF)=Main Channel Distance
X Axis Title(XS)=Station
BEGIN DESCRIPTION:
UNT 006 in La Jarita Watershed
END DESCRIPTION:
DSS Export Rating Curves= 0
DSS Export Rating Curve Sorted= 0
DSS Export Volume Flow Curves= 0
DXF OffsetX= 0
DXF OffsetY= 0
DXF ScaleX= 1
DXF ScaleY= 10

--- UNT 006 in La Jarita Watershed.p01 (plan) ---

Plan Title=Multiple Run
Short Identifier=Multiple
Geom File=g01
Flow File=f01
Subcritical Flow
K Sum by GR= 0
Std Step Tol= 0.01
Critical Tol= 0.01
Num of Std Step Trials= 20
Max Error Tol= 0.3
Flow Tol Ratio= 0.001
Split Flow NTrial= 30
Split Flow Tol= 0.02
Split Flow Ratio= 0.02
Log Output Level= 0
Friction Slope Method= 1
Unsteady Friction Slope Method= 2
Unsteady Bridges Friction Slope Method= 1
Parabolic Critical Depth
Global Vel Dist=  1 , 1 , 1
Global Log Level= 0
CheckData=True
Encroach Param= -1, 0, 0, 0
BEGIN DESCRIPTION:
Multiple Run
END DESCRIPTION:

--- UNT 006 in La Jarita Watershed.f01 (steady flow) ---

Flow Title=Multiple
Program Version=5.05
Number of Profiles= 7
Profile Names=10-year,25-year,50-year,1pct_min,100-year,1pct_plu,500-year
River Rch & RM=UNT 006 in La Ja,Reach-1         ,42125
     107     139     163      96     191     380     264
River Rch & RM=UNT 006 in La Ja,Reach-1         ,40064
     181     242     290     173     345     688     496
River Rch & RM=UNT 006 in La Ja,Reach-1         ,33430
     182     242     290     173     345     688     495
River Rch & RM=UNT 006 in La Ja,Reach-1         ,28575
     299     409     497     301     600    1197     888
River Rch & RM=UNT 006 in La Ja,Reach-1         ,19962
     412     571     701     428     853    1702    1284
River Rch & RM=UNT 006 in La Ja,Reach-1         ,8192
     543     762     944     581    1158    2311    1771
Boundary for River Rch & Prof#=UNT 006 in La Ja,Reach-1         , 1
Up Type= 0
Dn Type= 3
Dn Slope=0.0014
Boundary for River Rch & Prof#=UNT 006 in La Ja,Reach-1         , 2
Up Type= 0
Dn Type= 3
Dn Slope=0.0014
Boundary for River Rch & Prof#=UNT 006 in La Ja,Reach-1         , 3
Up Type= 0
Dn Type= 3
Dn Slope=0.0014
Boundary for River Rch & Prof#=UNT 006 in La Ja,Reach-1         , 4
Up Type= 0
Dn Type= 3
Dn Slope=0.0014
Boundary for River Rch & Prof#=UNT 006 in La Ja,Reach-1         , 5
Up Type= 0
Dn Type= 3
Dn Slope=0.0014
Boundary for River Rch & Prof#=UNT 006 in La Ja,Reach-1         , 6
Up Type= 0
Dn Type= 3
Dn Slope=0.0014
Boundary for River Rch & Prof#=UNT 006 in La Ja,Reach-1         , 7
Up Type= 0
Dn Type= 3
Dn Slope=0.0014
DSS Import GetInterval= 0
DSS Import GetPeak= 0
DSS Import FillOption= 0

--- UNT 006 in La Jarita Watershed.g01 (geometry) ---

Geom Title=Existing Conditions

River Reach=UNT 006 in La Ja,Reach-1
Reach XY= 30
      2107750.80     13418444.54      2105723.49     13418323.83
      2104863.48     13417241.49      2104730.80     13415954.54
      2103820.80     13414714.54      2108080.48     13411686.39
      2108440.80     13411514.54      2108940.80     13411894.54
      2109520.80     13410904.54      2110200.80     13410654.54
      2109926.55     13409049.19      2110824.99     13408725.84
      2111187.94     13407495.48      2111969.19     13407374.39
      2112870.23     13406561.89      2113439.25     13404797.48
      2114254.35     13404346.96      2115219.19     13402334.15
      2116700.80     13402294.54      2117120.80     13401694.54
      2118058.97     13401443.54      2120730.80     13401844.54
      2120840.80     13400774.54      2120270.80     13400854.54
      2120295.26     13399870.45      2119740.80     13399644.54
      2121440.80     13399024.54      2121800.80     13398504.54
      2121234.69     13398466.28      2120925.00     13397825.00

Type RM Length L Ch R = 1,42125,276,276,276
BEGIN DESCRIPTION:
UNT 006 in La Jarita Watershed 44.0
END DESCRIPTION:
XS GIS Cut Line= 3
      2107525.00     13417775.04      2107525.00     13418375.00
      2107675.00     13419725.03
#Sta/Elev= 30
  4410.5  341.43  4480.5  339.43  4530.5  335.88  4590.5  333.99  4630.5  331.58
  4690.5  329.27  4790.5  327.11  4850.5  326.71  4870.5  327.50  4910.5  326.31
  4970.5  326.70  4997.5  325.62  4998.0  324.82  5003.0  324.82  5003.5  325.62
  5131.2  327.18  5161.4  328.95  5181.5  330.83  5241.9  333.50  5282.1  334.14
  5362.6  333.86  5453.2  336.14  5503.5  335.48  5563.8  335.75  5905.9  338.51
  5926.1  339.23  6077.0  340.10  6157.5  339.96  6268.2  341.45  6368.8  341.47
#Mann=3,-1,0
  4410.5     0.1       0  4997.5    0.07       0  5003.5     0.1       0
Bank Sta=4997.5,5003.5
Exp/Cntr=0.3,0.1

Type RM Length L Ch R = 1,41849,307,307,307
BEGIN DESCRIPTION:
UNT 006 in La Jarita Watershed 43.0
END DESCRIPTION:
XS GIS Cut Line= 3
      2107474.99     13417725.04      2107275.00     13418425.00
      2107575.01     13419325.04
#Sta/Elev= 30
  4252.0  341.98  4293.6  341.87  4341.7  339.97  4380.7  339.10  4439.2  336.18
  4521.1  333.44  4526.3  333.63  4616.0  329.17  4666.7  327.80  4751.2  326.03
  4783.7  325.96  4844.8  324.93  4938.4  324.73  4990.5  325.19  5019.1  324.39
  5019.6  323.59  5024.6  323.59  5025.1  324.39  5053.8  325.69  5180.2  327.17
  5306.7  329.42  5443.8  334.94  5485.9  335.08  5528.1  334.48  5612.4  335.69
  5675.7  336.01  5717.8  337.27  5749.5  337.59  5781.1  338.92  5928.7  340.20
#Mann=3,-1,0
  4252.0     0.1       0  5019.1    0.07       0  5025.1     0.1       0
Bank Sta=5019.1,5025.1
Exp/Cntr=0.3,0.1

Type RM Length L Ch R = 1,41542,282,282,282
BEGIN DESCRIPTION:
UNT 006 in La Jarita Watershed 42.0
END DESCRIPTION:
XS GIS Cut Line= 3
      2107325.00     13417925.01      2107025.00     13418425.00
      2107424.99     13419224.99
#Sta/Elev= 30
  4464.1  338.78  4471.9  338.29  4477.7  338.60  4508.8  336.51  4572.9  334.09
  4588.5  332.59  4646.8  329.18  4674.0  328.35  4917.0  324.09  4981.1  323.46
  5033.6  323.81  5041.3  323.03  5041.8  322.23  5046.8  322.23  5047.3  323.03
  5069.5  323.65  5105.9  323.39  5145.0  324.54  5167.4  324.28  5234.5  324.99
  5382.6  327.66  5435.7  329.22  5553.1  330.78  5681.7  334.06  5709.6  334.16
  5785.1  335.98  5807.4  337.00  5821.4  337.04  5838.2  338.08  5941.6  339.89
#Mann=3,-1,0
  4464.1     0.1       0  5041.3    0.07       0  5047.3     0.1       0
Bank Sta=5041.3,5047.3
Exp/Cntr=0.3,0.1

Type RM Length L Ch R = 1,41260,347,347,347
BEGIN DESCRIPTION:
UNT 006 in La Jarita Watershed 41.0
END DESCRIPTION:
XS GIS Cut Line= 3
      2107025.02     13417924.97      2106775.00     13418375.00
      2107375.01     13419275.01
#Sta/Elev= 30
  4461.7  337.42  4475.5  337.53  4535.0  336.05  4551.0  334.63  4600.2  333.54
  4770.6  324.37  4827.8  323.27  4850.7  321.89  4881.6  321.84  4909.0  322.50
  4990.0  321.83  4996.1  321.27  4996.6  320.47  5001.6  320.47  5002.1  321.27
  5041.1  322.54  5071.2  321.97  5098.2  322.90  5179.3  323.07  5236.4  324.10
  5395.7  325.57  5458.8  328.28  5467.8  328.14  5517.4  331.32  5560.9  332.35
  5669.1  334.45  5855.4  336.08  5900.4  338.02  5950.0  339.27  6058.2  340.67
#Mann=3,-1,0
  4461.7     0.1       0  4996.1    0.07       0  5002.1     0.1       0
Bank Sta=4996.1,5002.1
Exp/Cntr=0.3,0.1

Type RM Length L Ch R = 1,40913,849,849,849
BEGIN DESCRIPTION:
Mapping XS 4920b53d
END DESCRIPTION:
XS GIS Cut Line= 3
      2107041.41     13417646.94      2106473.70     13418292.78
      2106306.73     13420011.40
#Sta/Elev= 30
  4108.2  344.28  4395.0  345.09  4415.9  343.78  4458.6  337.59  4501.3  333.04
  4600.0  325.62  4642.7  323.66  4728.0  321.36  4791.6  320.51  5037.7  320.26
  5038.2  319.46  5043.2  319.46  5043.7  320.26  5090.9  321.05  5241.6  321.07
  5311.7  322.27  5362.2  322.10  5392.3  323.07  5583.2  323.98  5627.6  324.79
  5713.8  329.16  5764.0  328.92  5804.2  331.63  5864.5  332.80  5933.5  335.18
  6055.4  336.12  6351.3  340.20  6397.0  341.43  6577.9  343.24  6694.8  343.59
#Mann=3,-1,0
  4108.2     0.1       0  5037.7    0.07       0  5043.7     0.1       0
Bank Sta=5037.7,5043.7
Exp/Cntr=0.3,0.1

Type RM Length L Ch R = 1,40064,319,319,319
BEGIN DESCRIPTION:
UNT 006 in La Jarita Watershed 40.0
END DESCRIPTION:
XS GIS Cut Line= 3
      2106887.73     13417659.98      2105575.00     13418325.00
      2105275.00     13419825.02
#Sta/Elev= 30
  3638.3  344.34  3742.3  344.39  3770.7  343.48  3809.5  340.23  3820.8  338.45
  3843.1  336.09  3910.4  331.28  4022.5  324.18  4121.5  319.93  4224.3  318.77
  4403.6  318.44  4461.2  317.17  4500.1  317.57  4589.2  316.82  4639.4  317.27
  4796.0  315.96  4856.5  316.10  5104.1  314.74  5104.6  313.94  5109.6  313.94
  5110.1  314.74  5466.8  316.79  5670.8  319.41  5762.5  319.77  6252.1  324.56
  6354.0  326.67  6394.8  328.37  6527.4  335.57  6609.0  338.83  6639.6  339.52
#Mann=3,-1,0
  3638.3     0.1       0  5104.1    0.07       0  5110.1     0.1       0
Bank Sta=5104.1,5110.1
Exp/Cntr=0.3,0.1

Type RM Length L Ch R = 1,39745,287,287,287
BEGIN DESCRIPTION:
UNT 006 in La Jarita Watershed 39.0
END DESCRIPTION:
XS GIS Cut Line= 3
      2106848.68     13417610.50      2105375.00     13418075.00
      2104775.00     13419575.00
#Sta/Elev= 30
  3529.1  344.51  3553.9  344.94  3669.3  344.11  3694.6  342.56  3727.0  336.82
  3732.2  337.02  3759.3  333.11  3791.7  329.90  3926.4  320.67  3958.7  318.92
  3991.1  318.32  4287.6  316.77  4330.4  317.08  4853.4  313.83  5280.2  313.87
  5301.4  313.30  5301.9  312.50  5307.0  312.50  5307.5  313.30  5382.6  314.43
  5872.6  316.35  5945.3  317.46  6043.6  317.86  6151.3  319.47  6195.7  321.15
  6291.3  319.97  6334.4  320.46  6572.7  326.00  6614.4  328.00  6689.8  333.45
#Mann=3,-1,0
  3529.1     0.1       0  5301.4    0.07       0  5307.5     0.1       0
Bank Sta=5301.4,5307.5
Exp/Cntr=0.3,0.1

Type RM Length L Ch R = 1,39458,371,371,371
BEGIN DESCRIPTION:
UNT 006 in La Jarita Watershed 38.0
END DESCRIPTION:
XS GIS Cut Line= 3
      2107226.32     13417464.65      2105275.00     13417825.00
      2104274.99     13419825.02
#Sta/Elev= 30
  3023.3  337.65  3051.4  337.56  3056.5  338.88  3065.3  339.02  3104.4  338.69
  3109.4  339.81  3215.4  337.74  3268.3  339.27  3326.3  342.86  3451.7  345.70
  3553.4  339.66  3712.3  325.50  3770.3  322.65  3823.3  318.14  3919.5  316.66
  4031.4  316.94  4661.9  313.00  5002.0  312.27  5002.5  311.47  5007.6  311.47
  5008.1  312.27  5231.2  313.50  5343.0  312.82  5879.7  314.29  6066.9  316.15
  6184.3  316.03  6268.2  317.64  6438.7  316.84  7020.1  325.62  7243.7  327.82
#Mann=3,-1,0
  3023.3     0.1       0  5002.0    0.07       0  5008.1     0.1       0
Bank Sta=5002,5008.1
Exp/Cntr=0.3,0.1

Type RM Length L Ch R = 1,39087,223,223,223
BEGIN DESCRIPTION:
UNT 006 in La Jarita Watershed 37.0
END DESCRIPTION:
XS GIS Cut Line= 3
      2107200.29     13417321.42      2105175.00     13417525.00
      2103924.99     13420025.01
#Sta/Elev= 30
  2964.5  329.62  3040.2  328.29  3140.7  333.46  3190.9  337.41  3271.3  338.83
  3291.4  338.31  3348.5  333.85  3371.8  333.48  3549.0  322.74  3554.0  323.16
  3649.2  317.75  3749.4  315.07  4944.3  311.33  4944.8  310.53  4949.9  310.53
  4950.4  311.33  5371.7  313.11  6051.0  313.49  6193.5  314.92  6266.2  314.00
  6400.3  314.81  6506.6  317.88  6587.6  315.38  6735.7  316.24  7222.1  323.25
  7280.8  322.93  7451.3  324.86  7579.9  327.94  7697.3  333.78  7795.1  335.87
#Mann=3,-1,0
  2964.5     0.1       0  4944.3    0.07       0  4950.4     0.1       0
Bank Sta=4944.3,4950.4
Exp/Cntr=0.3,0.1

Type RM Length L Ch R = 1,38864,305,305,305
BEGIN DESCRIPTION:
Mapping XS 61280038
END DESCRIPTION:
XS GIS Cut Line= 4
      2106752.28     13417354.89      2105637.72     13417073.65
      2104773.14     13417490.31      2104409.29     13418166.04
#Sta/Elev= 30
  3180.6  330.57  3250.0  324.68  3279.0  323.64  3373.7  317.35  3456.3  314.69
  3538.8  313.73  3612.7  313.50  3662.5  312.70  3703.8  313.10  3859.1  312.70
  4240.1  310.95  4528.2  310.83  4641.3  311.49  4663.9  310.87  4777.0  311.69
  5036.9  311.22  5050.9  310.82  5051.4  310.02  5056.5  310.02  5057.0  310.82
  5099.1  311.47  5195.2  311.02  5289.5  311.83  5386.3  311.55  5512.0  312.36
  5971.2  313.31  5993.1  313.71  6036.9  316.59  6053.1  316.81  6057.3  317.50
#Mann=3,-1,0
  3180.6     0.1       0  5050.9    0.07       0  5057.0     0.1       0
Bank Sta=5050.9,5057
Exp/Cntr=0.3,0.1

Type RM Length L Ch R = 1,38559,352,352,352
BEGIN DESCRIPTION:
Mapping XS c957f9bc
END DESCRIPTION:
XS GIS Cut Line= 4
      2106778.32     13417334.05      2105460.64     13416813.23
      2104559.60     13417323.65      2104330.44     13418177.80
#Sta/Elev= 30
  2876.5  330.29  2970.3  323.55  3019.0  321.17  3054.1  317.86  3078.5  316.27
  3192.0  313.61  3270.5  313.47  3324.6  312.36  3486.8  311.78  3546.7  312.21
  3933.8  310.43  4495.3  310.85  4548.8  310.73  4583.1  309.73  4583.6  308.93
  4589.0  308.93  4589.5  309.73  4629.6  310.80  4931.1  310.09  5207.8  311.71
  5288.3  311.36  5366.3  312.06  5609.9  312.04  5692.7  312.83  5765.2  312.33
  6100.5  313.14  6140.5  314.39  6175.3  317.40  6200.1  318.82  6213.3  318.55
#Mann=3,-1,0
  2876.5     0.1       0  4583.1    0.07       0  4589.5     0.1       0
Bank Sta=4583.1,4589.5
Exp/Cntr=0.3,0.1

Type RM Length L Ch R = 1,38207,374,374,374
BEGIN DESCRIPTION:
Mapping XS 94a434f3
END DESCRIPTION:
XS GIS Cut Line= 4
      2106658.52     13417261.12      2105481.47     13416641.35
      2104398.14     13416933.02      2104221.27     13418181.50
#Sta/Elev= 30
  2975.2  320.36  3025.3  316.26  3080.1  314.58  3278.4  312.14  3316.8  312.33
  3410.6  311.42  3454.6  311.87  3515.1  311.10  3597.6  311.30  3795.9  310.15
  4004.9  310.52  4120.7  310.01  4247.3  310.88  4458.2  310.85  4873.7  309.08
  4874.2  308.28  4879.6  308.28  4880.1  309.08  5171.7  310.12  5254.6  311.36
  5307.7  310.93  5449.6  311.83  5641.4  311.71  5669.4  312.27  6200.2  313.07
  6520.1  312.93  6626.1  314.40  6671.6  318.86  6681.7  318.67  6688.3  317.85
#Mann=5,-1,0
  2975.2     0.1       0  4873.7    0.07       0  4880.1     0.1       0
  5307.7    0.05       0  5669.4     0.1       0
Bank Sta=4873.7,4880.1
Exp/Cntr=0.3,0.1

Type RM Length L Ch R = 1,37833,456,456,456
BEGIN DESCRIPTION:
Mapping XS 31e0292b
END DESCRIPTION:
XS GIS Cut Line= 4
      2105642.97     13416641.38      2105247.10     13416365.31
      2104293.97     13416672.60      2104132.51     13418094.50
#Sta/Elev= 30
  4122.0  310.39  4176.4  310.42  4241.1  310.92  4708.9  309.57  4915.0  308.55
  4964.1  308.82  5002.7  308.35  5003.2  307.55  5008.7  307.55  5009.2  308.35
  5216.9  309.38  5267.6  309.77  5289.8  309.40  5321.3  310.08  5374.3  310.09
  5447.4  310.88  5809.8  311.47  5870.1  311.94  5940.6  311.67  5955.7  312.03
  5970.8  312.42  6192.2  312.03  6363.3  312.70  6433.7  312.33  6484.1  313.07
  6534.4  312.53  6635.0  313.07  6866.5  312.34  6977.2  313.27  7037.1  313.20
#Mann=7,-1,0
  4122.0     0.1       0  4176.4    0.05       0  4708.9     0.1       0
  5002.7    0.07       0  5009.2     0.1       0  5216.9    0.05       0
  5955.7     0.1       0
Bank Sta=5002.7,5009.2
Exp/Cntr=0.3,0.1

Type RM Length L Ch R = 1,37377,301,301,301
BEGIN DESCRIPTION:
Mapping XS ca227102
END DESCRIPTION:
XS GIS Cut Line= 4
      2105622.09     13416589.26      2104997.10     13416016.35
      2104137.72     13416245.52      2104064.88     13417551.44
#Sta/Elev= 30
  3886.9  310.31  4022.2  310.91  4100.0  310.31  4213.3  310.40  4369.4  309.43
  4453.8  309.46  4581.5  308.43  4822.8  308.47  5147.6  307.31  5148.1  306.51
  5153.6  306.51  5154.1  307.31  5181.9  307.97  5275.1  307.90  5420.0  309.53
  5486.8  309.56  5521.7  310.22  6062.0  311.28  6253.0  311.90  6384.8  311.81
  6414.9  312.34  6464.9  311.97  6565.1  312.53  6615.2  312.10  6645.2  312.58
  6745.4  312.35  6775.4  312.81  6865.6  312.54  6925.6  313.39  6932.1  312.84
#Mann=6,-1,0
  3886.9    0.05       0  4822.8     0.1       0  5147.6    0.07       0
  5154.1     0.1       0  6062.0    0.05       0  6253.0     0.1       0
Bank Sta=5147.6,5154.1
Exp/Cntr=0.3,0.1

Type RM Length L Ch R = 1,37076,262,262,262
BEGIN DESCRIPTION:
Mapping XS 7860d87f
END DESCRIPTION:
XS GIS Cut Line= 4
      2105632.54     13416537.21      2104835.64     13415750.73
      2104106.47     13416031.98      2103997.10     13417495.53
#Sta/Elev= 30
  3657.1  310.74  4010.5  310.27  4038.8  309.58  4236.8  308.85  4272.1  308.20
  4307.5  308.72  4371.1  308.15  4420.6  308.67  4554.9  308.52  4611.5  307.62
  4717.6  307.98  4755.3  307.52  4856.3  307.11  4926.1  306.96  5010.0  306.62
  5010.5  305.82  5016.0  305.82  5016.5  306.62  5152.6  307.46  5196.2  306.92
  5227.6  307.76  5439.1  309.94  5645.8  310.37  5691.7  309.95  6185.0  311.64
  6473.8  311.64  6604.2  312.39  6634.3  311.89  6844.9  312.87  7025.9  312.83
#Mann=6,-1,0
  3657.1    0.05       0  4755.3     0.1       0  4856.3    0.05       0
  4926.1     0.1       0  5010.0    0.07       0  5016.5     0.1       0
Bank Sta=5010,5016.5
Exp/Cntr=0.3,0.1

Type RM Length L Ch R = 1,36814,394,394,394
BEGIN DESCRIPTION:
Mapping XS bce27fe4
END DESCRIPTION:
XS GIS Cut Line= 4
      2105554.40     13416412.19      2104773.14     13415547.60
      2104059.60     13415771.56      2103976.26     13417235.15
#Sta/Elev= 30
  3484.3  310.73  3552.6  310.54  3581.0  310.98  3664.8  310.28  3878.4  308.29
  3974.3  308.21  4055.5  307.80  4104.8  308.22  4204.2  307.30  4281.9  307.76
  4441.6  307.19  4600.3  306.85  4642.9  306.26  4703.3  306.56  4957.5  306.20
  4986.6  305.64  4987.1  304.84  4992.6  304.84  4993.1  305.64  5014.7  306.12
  5077.4  305.99  5130.0  307.03  5254.5  307.76  5292.1  308.44  5401.7  308.18
  5631.3  309.78  5791.5  309.78  6382.5  311.87  6797.9  311.84  6863.4  312.51
#Mann=8,-1,0
  3484.3    0.05       0  3664.8     0.1       0  3974.3    0.05       0
  4441.6     0.1       0  4703.3    0.05       0  4986.6   0.035       0
  4993.1    0.05       0  5014.7     0.1       0
Bank Sta=4986.6,4993.1
Exp/Cntr=0.3,0.1

Type RM Length L Ch R = 1,36420,313,313,313
BEGIN DESCRIPTION:
Mapping XS b6a83471
END DESCRIPTION:
XS GIS Cut Line= 4
      2105455.45     13416235.13      2104679.39     13415313.23
      2103892.93     13415469.48      2103913.77     13417177.86
#Sta/Elev= 30
  3286.6  309.82  3556.4  307.59  3605.3  307.69  3699.9  307.49  3783.5  306.77
  4097.9  306.69  4453.4  306.20  4634.7  306.65  4830.9  306.25  5043.4  304.42
  5043.9  303.62  5049.4  303.62  5049.9  304.42  5158.8  305.57  5188.9  305.09
  5299.0  305.07  5559.0  307.45  5709.0  307.69  5749.0  308.29  5809.1  308.10
  5873.5  308.85  6079.1  309.45  6189.1  310.39  6219.1  310.06  6239.1  310.50
  6499.1  311.35  6549.1  311.02  6619.1  311.88  6729.1  311.55  7002.0  311.93
#Mann=9,-1,0
  3286.6     0.1       0  3556.4    0.05       0  3605.3     0.1       0
  3699.9    0.05       0  4097.9     0.1       0  4453.4    0.05       0
  4634.7     0.1       0  5043.4    0.07       0  5049.9     0.1       0
Bank Sta=5043.4,5049.9
Exp/Cntr=0.3,0.1

Type RM Length L Ch R = 1,36107,430,430,430
BEGIN DESCRIPTION:
Mapping XS 6e3dfc0c
END DESCRIPTION:
XS GIS Cut Line= 4
      2105424.21     13416157.02      2104679.39     13415000.73
      2103637.72     13415281.98      2103835.55     13417150.86
#Sta/Elev= 30
  2957.8  308.98  3111.1  307.31  3262.3  307.48  3319.7  306.28  3421.9  305.87
  3501.1  305.83  3652.9  306.00  3900.8  305.96  3904.5  305.95  4072.6  305.96
  4160.8  305.68  4197.1  306.17  4290.8  305.28  4388.0  305.82  4640.3  306.18
  4928.2  304.94  4969.6  303.72  5011.0  303.64  5073.2  304.59  5212.9  304.59
  5266.3  303.63  5277.1  303.53  5277.6  302.73  5283.1  302.73  5283.6  303.53
  5404.5  303.65  6270.0  308.25  6482.5  309.91  7014.1  311.76  7291.5  311.94
#Mann=13,-1,0
  2957.8     0.1       0  3319.7    0.05       0  3421.9     0.1       0
  3501.1    0.05       0  3652.9     0.1       0  3900.8    0.05       0
  3904.5     0.1       0  4072.6    0.05       0  4388.0     0.1       0
  5266.3    0.05       0  5277.1    0.07       0  5283.6    0.05       0
  5404.5     0.1       0
Bank Sta=5277.1,5283.6
Exp/Cntr=0.3,0.1

Type RM Length L Ch R = 1,35677,473,473,473
BEGIN DESCRIPTION:
Mapping XS 9ead7796
END DESCRIPTION:
XS GIS Cut Line= 4
      2105497.12     13416214.30      2104778.35     13414880.94
      2103403.35     13414943.44      2103674.18     13417125.72
#Sta/Elev= 30
  2472.1  309.77  2539.5  309.41  2613.4  307.82  2766.7  307.54  2908.0  306.21
  2940.2  306.01  3151.3  305.31  3222.9  305.06  3438.7  305.53  3520.9  306.03
  3788.6  305.76  4010.2  304.51  4111.8  305.22  4430.7  305.44  4640.9  303.87
  4861.1  303.20  4971.2  303.91  5097.9  302.87  5098.4  302.07  5104.3  302.07
  5104.8  302.87  5135.4  303.16  5359.9  304.93  5538.7  303.75  5707.5  303.32
  5919.1  304.11  6815.9  310.30  7390.3  311.41  7451.5  312.13  7562.3  311.81
#Mann=11,-1,0
  2472.1     0.1       0  2908.0    0.05       0  2940.2     0.1       0
  3151.3    0.05       0  3222.9     0.1       0  3438.7    0.05       0
  4111.8     0.1       0  5097.9    0.07       0  5104.8     0.1       0
  5135.4    0.05       0  5538.7     0.1       0
Bank Sta=5097.9,5104.8
Exp/Cntr=0.3,0.1

Type RM Length L Ch R = 1,35204,637,637,637
BEGIN DESCRIPTION:
Mapping XS 69d5d619
END DESCRIPTION:
XS GIS Cut Line= 4
      2105543.98     13415615.32      2104903.35     13414802.81
      2103627.31     13414427.81      2102498.56     13414979.18
#Sta/Elev= 30
  3014.1  305.23  3184.2  304.04  3306.1  304.61  3381.2  304.37  3498.4  305.25
  3625.8  305.53  3840.1  304.73  4009.9  305.08  4166.0  304.48  4193.0  304.94
  4260.7  304.78  4443.1  304.74  4559.1  303.82  4599.5  304.18  4764.6  303.14
  4797.5  303.43  4933.0  302.71  4964.3  303.09  5087.5  302.69  5088.0  301.89
  5093.9  301.89  5094.4  302.69  5338.5  303.87  5362.2  303.75  5475.4  304.22
  5526.0  305.22  5593.6  305.04  5691.0  305.64  6450.0  306.62  6635.0  307.07
#Mann=9,-1,0
  3014.1     0.1       0  3381.2    0.05       0  4260.7     0.1       0
  5087.5    0.07       0  5094.4     0.1       0  5338.5    0.05       0
  5362.2     0.1       0  5691.0    0.05       0  6450.0     0.1       0
Bank Sta=5087.5,5094.4
Exp/Cntr=0.3,0.1

Type RM Length L Ch R = 1,34567,555,555,555
BEGIN DESCRIPTION:
Mapping XS 0d31bc63
END DESCRIPTION:
XS GIS Cut Line= 4
      2105314.79     13415255.90      2105007.52     13414547.60
      2104174.18     13414047.60      2102596.02     13414839.29
#Sta/Elev= 30
  3637.7  304.83  3845.5  304.62  3874.5  304.96  4020.2  304.36  4329.5  304.63
  4471.0  304.34  4529.3  303.64  4559.5  304.05  4699.8  303.49  4866.6  303.34
  5017.3  302.55  5063.0  302.83  5108.9  302.16  5109.4  301.36  5115.4  301.36
  5115.9  302.16  5142.7  302.36  5328.4  302.97  5425.4  303.42  5481.6  302.91
  5648.5  303.38  5788.7  303.27  5861.8  303.81  5922.7  303.48  6309.3  305.64
  6376.4  305.55  6408.6  306.12  6445.3  305.83  6986.1  306.15  7147.2  306.72
#Mann=10,-1,0
  3637.7    0.05       0  4699.8     0.1       0  5017.3    0.05       0
  5108.9    0.07       0  5115.9    0.05       0  5142.7     0.1       0
  5328.4    0.05       0  5648.5     0.1       0  6445.3    0.05       0
  6986.1     0.1       0
Bank Sta=5108.9,5115.9
Exp/Cntr=0.3,0.1

Type RM Length L Ch R = 1,34012,344,344,344
BEGIN DESCRIPTION:
Mapping XS 1721ae3a
END DESCRIPTION:
XS GIS Cut Line= 4
      2105340.85     13415141.34      2105226.27     13414360.10
      2104668.97     13413630.94      2103064.81     13414245.52
#Sta/Elev= 30
  3774.5  304.39  3801.1  304.75  3882.0  303.85  3932.5  303.99  3962.8  303.58
  3993.2  304.06  4094.2  303.75  4225.6  304.38  4448.0  304.05  4775.1  302.50
  4874.9  302.62  5014.7  301.62  5015.2  300.82  5021.2  300.82  5021.7  301.62
  5089.6  301.77  5282.1  303.38  5367.3  303.22  5496.8  303.74  5559.4  303.33
  5594.8  303.75  5759.0  303.60  6192.9  304.54  6332.1  304.10  6546.5  304.27
  6631.9  305.00  6781.9  304.95  6880.2  305.52  6934.9  305.05  7199.7  306.01
#Mann=4,-1,0
  3774.5    0.05       0  5014.7    0.03       0  5021.7    0.05       0
  5089.6     0.1       0
Bank Sta=5014.7,5021.7
Exp/Cntr=0.3,0.1

Type RM Length L Ch R = 1,33668,238,238,238
BEGIN DESCRIPTION:
Mapping XS 4cf73d39
END DESCRIPTION:
XS GIS Cut Line= 4
      2105356.48     13414964.27      2105533.56     13414235.10
      2105038.77     13413537.19      2104085.63     13413771.56
#Sta/Elev= 30
  3680.6  303.62  3762.2  303.39  3793.0  303.78  3875.4  303.19  4034.7  303.97
  4060.6  303.45  4081.6  303.88  4334.9  303.19  4554.8  302.73  4686.2  302.52
  4774.3  301.62  4846.6  301.57  4870.4  301.32  4870.9  300.52  4876.9  300.52
  4877.4  301.32  4916.1  301.58  4974.8  301.42  5025.3  302.15  5054.8  301.86
  5111.4  302.92  5240.1  303.63  5268.9  303.25  5509.7  303.19  5681.7  303.74
  5883.5  303.44  5980.3  304.16  6054.8  303.90  6132.7  304.37  6268.0  304.17
#Mann=8,-1,0
  3680.6    0.05       0  4334.9     0.1       0  4554.8    0.05       0
  4686.2     0.1       0  4846.6    0.05       0  4870.4    0.07       0
  4877.4    0.05       0  4916.1     0.1       0
Bank Sta=4870.4,4877.4
Exp/Cntr=0.3,0.1

Type RM Length L Ch R = 1,33430,34,34,34
BEGIN DESCRIPTION:
Mapping XS d865d501
END DESCRIPTION:
XS GIS Cut Line= 4
      2105408.56     13414953.84      2105710.64     13414042.40
      2105148.14     13413328.85      2103653.32     13413896.57
#Sta/Elev= 30
  3471.8  303.30  3715.0  303.50  3818.2  303.26  3839.3  303.70  4028.1  302.73
  4060.5  303.11  4169.1  302.69  4297.3  302.63  4576.8  302.80  4632.4  302.10
  4694.9  301.87  4735.0  301.49  4879.5  301.16  4880.0  300.36  4886.0  300.36
  4886.5  301.16  5061.0  302.57  5089.9  302.36  5167.2  303.40  5354.7  302.93
  5396.1  303.45  5450.9  303.05  5525.8  303.48  5566.2  303.11  5826.7  303.60
  5961.2  303.30  6146.2  304.12  6263.9  303.86  6392.3  304.43  6939.6  304.79
#Mann=10,-1,0
  3471.8    0.05       0  3715.0     0.1       0  4028.1    0.05       0
  4169.1     0.1       0  4297.3    0.05       0  4632.4     0.1       0
  4694.9    0.05       0  4735.0     0.1       0  4879.5    0.07       0
  4886.5     0.1       0
Bank Sta=4879.5,4886.5
Exp/Cntr=0.3,0.1

Type RM Length L Ch R = 1,33396,27,27,27
BEGIN DESCRIPTION:
Mapping XS cc32e5ff
END DESCRIPTION:
XS GIS Cut Line= 6
      2105534.43     13414642.21      2105616.89     13413665.66
      2105859.95     13413292.40      2105438.94     13413635.28
      2105130.78     13413288.06      2103863.42     13413804.55
#Sta/Elev= 30
  2854.6  303.11  3041.5  302.86  3230.4  302.78  3324.6  302.52  3686.1  302.05
  3859.3  301.83  3900.2  300.54  3922.7  301.83  3958.9  300.38  3980.0  302.20
  3995.1  300.37  4002.5  301.71  4018.5  299.94  4042.5  299.60  4047.9  301.22
  4071.9  298.33  4077.3  299.28  4095.9  297.70  4266.1  298.45  4357.2  299.60
  4502.1  298.36  4557.5  298.65  4603.7  297.15  4604.2  296.35  4610.8  297.15
  4644.9  297.92  4720.5  298.16  4784.0  300.66  5159.4  303.15  6748.6  304.44
#Mann=13,-1,0
  2854.6     0.1       0  3041.5    0.05       0  3230.4     0.1       0
  3324.6    0.05       0  3686.1     0.1       0  3859.3    0.07       0
  3900.2     0.1       0  4095.9    0.07       0  4266.1     0.1       0
  4502.1    0.07       0  4603.7    0.07       0  4610.8    0.07       0
  4644.9     0.1       0
Bank Sta=4603.7,4610.8
Exp/Cntr=0.3,0.1

Type RM Length L Ch R = 1,33369,500,500,500
BEGIN DESCRIPTION:
Mapping XS b6449aed
END DESCRIPTION:
XS GIS Cut Line= 6
      2105559.61     13414662.15      2105648.14     13413740.31
      2105861.68     13413240.31      2105424.18     13413578.85
      2105122.10     13413245.52      2103794.00     13413797.59
#Sta/Elev= 30
  2806.0  303.18  2960.1  302.80  3206.8  302.58  3268.0  302.39  3658.3  302.40
  3777.5  301.46  3778.0  300.66  3784.0  300.66  3784.6  301.46  3850.0  304.44
  4037.5  306.01  4319.6  303.02  4365.9  303.60  4394.6  303.97  4449.8  303.17
  4478.6  304.01  4484.3  302.95  4500.5  304.36  4506.2  303.39  4522.4  305.08
  4528.1  304.52  4544.3  305.67  4615.3  305.02  4636.0  305.84  4700.5  304.74
  4884.1  304.12  4954.8  301.82  5179.7  303.16  5682.2  302.84  6853.3  304.63
#Mann=11,-1,0
  2806.0     0.1       0  2960.1    0.05       0  3206.8     0.1       0
  3268.0    0.05       0  3658.3     0.1       0  3777.5    0.07       0
  3784.6     0.1       0  4365.9    0.05       0  4394.6     0.1       0
  4615.3    0.07       0  4700.5     0.1       0
Bank Sta=3777.5,3784.6
Exp/Cntr=0.3,0.1

Type RM Length L Ch R = 1,32869,320,320,320
BEGIN DESCRIPTION:
Mapping XS a7c6c210
END DESCRIPTION:
XS GIS Cut Line= 6
      2105570.01     13414667.41      2105898.14     13413209.06
      2105648.14     13413193.44      2105382.52     13413479.90
      2105116.89     13413162.19      2103726.29     13413802.80
#Sta/Elev= 30
  3190.9  303.20  3321.5  302.82  3607.5  302.56  3631.2  302.51  4048.3  302.75
  4181.7  301.59  4439.8  301.96  4469.4  301.47  4490.3  301.96  4684.8  300.52
  4722.6  301.03  4745.4  300.15  4745.9  299.35  4751.9  299.35  4752.5  300.15
  4771.4  300.67  4796.9  301.44  4833.0  301.35  4910.7  300.60  5092.5  301.82
  5120.8  301.36  5446.3  302.01  5567.1  303.27  5764.9  302.62  6200.8  302.68
  6390.0  303.57  6682.0  303.55  6788.6  304.35  6968.5  303.97  7403.7  305.03
#Mann=9,-1,0
  3190.9     0.1       0  3321.5    0.05       0  3607.5     0.1       0
  3631.2    0.05       0  4048.3     0.1       0  4745.4    0.07       0
  4752.5     0.1       0  4771.4    0.05       0  4833.0     0.1       0
Bank Sta=4745.4,4752.5
Exp/Cntr=0.3,0.1

Type RM Length L Ch R = 1,32549,342,342,342
BEGIN DESCRIPTION:
Mapping XS 095186a9
END DESCRIPTION:
XS GIS Cut Line= 4
      2105798.73     13414110.42      2106173.75     13413323.93
      2105902.92     13412964.56      2104413.33     13413303.10
#Sta/Elev= 30
  3827.1  302.38  3857.0  302.28  3874.2  302.76  3970.5  302.18  3999.3  302.69
  4020.7  302.22  4129.4  302.57  4180.3  301.96  4339.2  302.20  4690.7  301.46
  4856.7  299.82  4871.2  299.64  4871.7  298.84  4877.7  298.84  4878.3  299.64
  4918.4  300.32  5015.4  300.27  5145.0  301.79  5177.6  301.38  5207.8  301.85
  5300.1  302.01  5433.4  301.71  5505.2  302.33  5864.1  302.72  6069.2  302.24
  6202.6  302.99  6294.8  302.48  6541.0  303.11  6574.3  303.53  6676.0  303.44
#Mann=6,-1,0
  3827.1    0.05       0  4020.7     0.1       0  4856.7    0.05       0
  4871.2    0.03       0  4878.3    0.05       0  5015.4     0.1       0
Bank Sta=4871.2,4878.3
Exp/Cntr=0.3,0.1

Type RM Length L Ch R = 1,32207,171,171,171
BEGIN DESCRIPTION:
Mapping XS c563d469
END DESCRIPTION:
XS GIS Cut Line= 4
      2105845.61     13414089.59      2106439.37     13413136.43
      2106106.04     13412740.60      2104444.61     13413245.80
#Sta/Elev= 30
  3621.2  302.17  3646.4  302.52  3774.3  302.01  3898.9  302.31  3921.1  301.78
  3980.1  302.09  4015.4  301.64  4097.2  301.91  4168.6  301.40  4197.5  301.82
  4349.7  301.16  4501.9  301.25  4553.8  301.81  4690.7  301.45  4721.4  301.91
  4833.7  301.56  4966.8  300.01  5064.2  299.26  5064.7  298.46  5070.8  298.46
  5071.3  299.26  5165.4  299.96  5216.7  300.80  5428.1  301.89  5772.4  301.33
  5942.0  302.19  5980.1  301.81  6286.3  302.58  6788.8  302.54  6998.2  303.64
#Mann=6,-1,0
  3621.2    0.05       0  3774.3     0.1       0  4966.8    0.05       0
  5064.2    0.03       0  5071.3    0.05       0  5165.4     0.1       0
Bank Sta=5064.2,5071.3
Exp/Cntr=0.3,0.1

Type RM Length L Ch R = 1,32036,247,247,247
BEGIN DESCRIPTION:
Mapping XS fcfc0f15
END DESCRIPTION:
XS GIS Cut Line= 4
      2106194.61     13413631.19      2106632.08     13413053.10
      2106132.08     13412558.31      2104845.62     13413027.06
#Sta/Elev= 30
  3942.8  301.56  3954.3  302.08  3975.6  301.37  4012.5  301.11  4312.1  301.50
  4462.0  301.05  4576.4  301.54  4618.0  301.07  4791.6  301.86  4855.3  301.64
  4984.3  299.88  5032.0  299.38  5106.3  299.38  5106.8  298.58  5112.9  298.58
  5113.4  299.38  5207.4  299.93  5343.2  301.53  5430.6  301.12  5485.2  301.55
  5517.0  301.01  5786.8  301.44  5804.5  301.11  5942.8  301.18  6168.2  301.95
  6357.9  301.82  6513.8  302.13  6544.3  302.60  6605.5  302.15  6740.4  302.56
#Mann=5,-1,0
  3942.8     0.1       0  4984.3    0.05       0  5106.3    0.03       0
  5113.4    0.05       0  5207.4     0.1       0
Bank Sta=5106.3,5113.4
Exp/Cntr=0.3,0.1

Type RM Length L Ch R = 1,31789,247,247,247
BEGIN DESCRIPTION:
Mapping XS e3c51141
END DESCRIPTION:
XS GIS Cut Line= 4
      2106246.70     13413631.19      2106788.33     13412928.10
      2106361.25     13412381.23      2104898.82     13412912.07
#Sta/Elev= 30
  3762.6  301.40  4000.7  300.99  4108.5  301.40  4150.2  300.87  4193.7  301.22
  4278.8  300.92  4357.7  301.31  4515.2  301.16  4704.8  302.10  4875.5  300.95
  4947.6  299.92  4975.0  299.44  5099.9  298.92  5100.4  298.12  5106.5  298.12
  5107.0  298.92  5267.5  300.72  5301.5  300.72  5368.2  301.24  5429.0  301.05
  5510.2  301.50  5627.3  300.92  5867.3  300.94  5953.8  301.34  5999.6  300.82
  6067.9  301.07  6225.4  301.21  6680.5  301.94  6733.7  302.51  6899.8  302.25
#Mann=9,-1,0
  3762.6     0.1       0  4947.6    0.05       0  5099.9    0.03       0
  5107.0    0.05       0  5267.5     0.1       0  5301.5    0.05       0
  5429.0     0.1       0  6067.9    0.05       0  6225.4     0.1       0
Bank Sta=5099.9,5107
Exp/Cntr=0.3,0.1

Type RM Length L Ch R = 1,31542,243,243,243
BEGIN DESCRIPTION:
Mapping XS 653a609c
END DESCRIPTION:
XS GIS Cut Line= 4
      2106268.37     13413629.05      2106915.07     13412934.61
      2106665.50     13412257.53      2105261.39     13412717.61
#Sta/Elev= 30
  3619.3  301.24  3740.0  300.95  3825.0  301.28  4001.9  300.74  4242.3  301.16
  4292.1  300.84  4390.8  301.45  4461.6  301.21  4613.8  301.66  4860.9  299.55
  4959.6  298.89  4960.1  298.09  4966.2  298.09  4966.7  298.89  5068.7  299.03
  5215.8  300.69  5547.4  301.20  5558.3  301.09  5732.2  301.39  5907.0  300.81
  6002.5  301.42  6071.4  300.65  6225.4  301.46  6257.2  300.33  6263.5  300.45
  6363.7  301.23  6501.5  300.76  6618.0  300.95  6658.4  301.48  6767.4  301.47
#Mann=9,-1,0
  3619.3     0.1       0  4860.9    0.05       0  4959.6    0.03       0
  4966.7    0.05       0  5547.4     0.1       0  5558.3    0.05       0
  5732.2     0.1       0  6263.5    0.05       0  6501.5     0.1       0
Bank Sta=4959.6,4966.7
Exp/Cntr=0.3,0.1

Type RM Length L Ch R = 1,31299,249,249,249
BEGIN DESCRIPTION:
Mapping XS e7097e25
END DESCRIPTION:
XS GIS Cut Line= 4
      2106450.68     13413479.30      2107101.70     13412849.98
      2106871.67     13412086.09      2105284.08     13412680.35
#Sta/Elev= 30
  3765.1  301.02  3933.9  300.83  3969.2  301.22  3997.4  300.76  4103.7  300.61
  4696.7  301.60  4777.7  301.26  4906.0  299.52  4953.2  298.72  5037.7  298.43
  5038.2  297.63  5044.3  297.63  5044.8  298.43  5304.2  300.64  5417.3  300.25
  5441.4  300.69  5468.3  300.30  5496.8  300.76  5590.6  300.65  5711.7  301.30
  5822.1  301.31  5902.3  300.75  5932.6  301.25  5977.3  300.81  6219.4  301.31
  6309.8  300.80  6531.1  301.18  6604.8  300.82  6932.9  301.13  7163.5  301.47
#Mann=7,-1,0
  3765.1     0.1       0  4906.0    0.05       0  5037.7    0.03       0
  5044.8    0.05       0  6309.8     0.1       0  6604.8    0.05       0
  6932.9     0.1       0
Bank Sta=5037.7,5044.8
Exp/Cntr=0.3,0.1

Type RM Length L Ch R = 1,31050,285,285,285
BEGIN DESCRIPTION:
Mapping XS c0a0a6ab
END DESCRIPTION:
XS GIS Cut Line= 4
      2106928.11     13413075.66      2107314.37     13412732.79
      2107084.34     13412060.05      2105691.15     13411903.80
#Sta/Elev= 30
  4151.3  301.20  4185.3  300.79  4220.4  301.12  4291.5  300.81  4510.6  301.45
  4631.0  300.50  4771.2  300.19  4895.2  298.87  4963.1  298.86  5016.8  298.35
  5017.3  297.55  5023.4  297.55  5023.9  298.35  5114.3  299.75  5130.5  299.49
  5183.3  300.09  5381.2  300.02  5438.5  300.45  5488.8  299.99  5643.6  300.56
  5831.9  300.32  5917.0  300.66  6059.3  300.06  6102.6  300.34  6354.2  300.26
  6457.9  300.98  6495.1  300.54  6633.1  300.92  6696.3  301.76  6780.7  301.24
#Mann=6,-1,0
  4151.3     0.1       0  4771.2    0.05       0  5016.8    0.03       0
  5023.9    0.05       0  5643.6     0.1       0  6059.3    0.05       0
Bank Sta=5016.8,5023.9
Exp/Cntr=0.3,0.1

Type RM Length L Ch R = 1,30765,177,177,177
BEGIN DESCRIPTION:
Mapping XS faf3d356
END DESCRIPTION:
XS GIS Cut Line= 4
      2107270.97     13412854.32      2107501.01     13412520.12
      2107314.37     13411908.14      2105899.75     13411721.54
#Sta/Elev= 30
  4277.2  300.86  4300.7  301.06  4373.5  300.28  4395.3  300.52  4505.1  299.87
  4523.8  299.76  4538.7  300.26  4616.5  299.41  4676.0  299.86  4761.4  298.99
  4914.7  298.53  4915.2  297.73  4921.3  297.73  4921.8  298.53  4929.1  298.84
  4990.6  298.70  5033.3  299.12  5132.3  299.98  5242.4  300.32  5274.1  299.92
  5594.4  300.09  5646.7  299.63  5695.6  300.08  5725.6  299.72  5796.2  299.98
  6276.3  299.63  6391.3  299.65  6534.8  300.28  6693.9  301.85  6749.6  302.01
#Mann=8,-1,0
  4277.2     0.1       0  4505.1    0.05       0  4914.7    0.07       0
  4921.8    0.05       0  4929.1     0.1       0  5033.3    0.05       0
  5646.7     0.1       0  6276.3    0.05       0
Bank Sta=4914.7,4921.8
Exp/Cntr=0.3,0.1

Type RM Length L Ch R = 1,30588,277,277,277
BEGIN DESCRIPTION:
Mapping XS 77c8cabd
END DESCRIPTION:
XS GIS Cut Line= 4
      2107427.23     13412680.70      2107600.83     13412402.93
      2107431.56     13411743.21      2106008.98     13411517.67
#Sta/Elev= 30
  4345.1  299.94  4352.1  299.87  4652.4  299.21  4711.5  299.75  4732.5  299.24
  4798.1  299.34  4902.0  298.48  4952.5  298.27  4953.0  297.47  4959.1  297.47
  4959.6  298.27  4981.1  298.35  5124.8  299.71  5154.7  299.49  5186.7  299.86
  5236.2  299.36  5331.3  299.86  5532.5  299.71  5573.0  300.04  5692.9  299.65
  5982.1  299.23  6018.5  299.37  6048.9  298.94  6099.5  299.31  6153.5  298.87
  6291.9  299.47  6397.1  299.20  6534.9  299.59  6602.8  300.17  6794.1  301.81
#Mann=10,-1,0
  4345.1     0.1       0  4352.1    0.05       0  4902.0     0.1       0
  4952.5    0.03       0  4959.6     0.1       0  4981.1    0.05       0
  5692.9     0.1       0  5982.1    0.05       0  6153.5     0.1       0
  6602.8    0.05       0
Bank Sta=4952.5,4959.6
Exp/Cntr=0.3,0.1

Type RM Length L Ch R = 1,30311,257,257,257
BEGIN DESCRIPTION:
Mapping XS 49010b05
END DESCRIPTION:
XS GIS Cut Line= 4
      2107448.91     13412698.09      2107804.83     13412146.85
      2107579.13     13411495.81      2106060.04     13411491.47
#Sta/Elev= 30
  4076.8  299.85  4086.7  299.86  4096.2  299.93  4144.0  299.60  4430.4  299.28
  4560.3  299.74  4716.7  299.22  4873.8  299.15  4904.9  298.28  4933.1  298.19
  4978.3  298.34  5006.5  297.77  5007.0  296.97  5013.1  296.97  5013.6  297.77
  5073.6  298.82  5148.8  298.88  5174.6  299.51  5354.8  299.43  5696.1  299.77
  5916.1  299.25  5956.1  298.66  6006.1  299.33  6089.4  299.13  6347.0  299.12
  6636.1  299.26  6766.1  300.10  6816.1  299.93  6864.0  300.61  6941.1  301.03
#Mann=12,-1,0
  4076.8     0.1       0  4086.7    0.05       0  4096.2     0.1       0
  4144.0    0.05       0  4716.7     0.1       0  4933.1    0.05       0
  5006.5    0.03       0  5013.6    0.05       0  5354.8     0.1       0
  6089.4    0.05       0  6347.0     0.1       0  6864.0    0.05       0
Bank Sta=5006.5,5013.6
Exp/Cntr=0.3,0.1

Type RM Length L Ch R = 1,30054,326,326,326
BEGIN DESCRIPTION:
Mapping XS 55df7237
END DESCRIPTION:
XS GIS Cut Line= 4
      2107470.60     13412693.76      2108030.52     13411977.58
      2107726.70     13411330.88      2106593.85     13410801.35
#Sta/Elev= 30
  3873.4  299.88  3883.9  299.88  3973.2  299.60  4217.1  299.32  4395.3  299.66
  4474.0  298.92  4544.6  299.17  4573.4  298.59  4602.4  298.89  4766.1  298.25
  4796.6  298.61  4873.2  298.23  4940.0  297.82  4969.7  298.15  5017.3  297.56
  5017.8  296.76  5023.9  296.76  5024.4  297.56  5112.1  298.77  5203.3  298.54
  5231.7  299.21  5251.7  298.98  5396.8  298.84  5465.3  298.31  5519.1  298.66
  5997.8  298.50  6204.7  298.78  6488.9  299.59  6705.5  301.97  6747.5  301.85
#Mann=10,-1,0
  3873.4    0.05       0  3883.9     0.1       0  3973.2    0.05       0
  4796.6     0.1       0  4873.2    0.05       0  5017.3    0.03       0
  5024.4    0.05       0  5251.7     0.1       0  5997.8    0.05       0
  6204.7     0.1       0
Bank Sta=5017.3,5024.4
Exp/Cntr=0.3,0.1

Type RM Length L Ch R = 1,29728,1153,1153,1153
BEGIN DESCRIPTION:
Mapping XS daf15fd4
END DESCRIPTION:
XS GIS Cut Line= 4
      2107560.50     13412595.31      2108294.84     13411772.43
      2108102.13     13411376.60      2106858.71     13410544.18
#Sta/Elev= 30
  3724.2  299.49  3855.3  299.81  3904.6  299.24  4110.3  299.74  4145.4  299.08
  4329.3  298.33  4606.0  298.48  4641.2  297.98  4690.5  298.31  4968.8  297.32
  4987.5  296.70  4988.0  295.90  4994.1  295.90  4994.7  296.70  4998.5  296.86
  5115.7  298.20  5367.6  298.36  5553.8  297.83  5640.9  298.32  5691.9  297.80
  5748.9  298.27  5836.0  297.87  5857.0  298.33  6001.1  297.91  6067.2  298.47
  6347.0  298.33  6391.4  299.15  6463.5  299.19  6649.6  301.69  6763.7  301.87
#Mann=4,-1,0
  3724.2    0.05       0  4987.5    0.07       0  4994.7    0.05       0
  4998.5     0.1       0
Bank Sta=4987.5,4994.7
Exp/Cntr=0.3,0.1

Type RM Length L Ch R = 1,28575,735,735,735
BEGIN DESCRIPTION:
Mapping XS fce7d4ab
END DESCRIPTION:
XS GIS Cut Line= 3
      2110164.61     13412756.78      2108586.51     13411267.22
      2107034.45     13410376.61
#Sta/Elev= 30
  3531.4  315.30  3567.8  312.20  3659.7  308.54  3666.9  307.68  3673.8  307.64
  3695.3  306.03  3772.9  302.95  3850.6  301.63  4183.2  297.62  4550.9  296.15
  4869.3  296.48  4935.7  295.08  4936.5  294.28  4943.7  294.28  4944.5  295.08
  4954.3  295.77  4982.6  295.12  5031.9  296.42  5173.5  297.09  5286.8  296.55
  5583.8  297.34  5968.4  297.27  6026.0  296.86  6378.3  297.75  6561.0  297.31
  6759.5  297.77  6787.0  297.34  6877.4  298.00  7167.9  298.37  7490.9  301.19
#Mann=3,-1,0
  3531.4     0.1       0  4935.7    0.07       0  4944.5     0.1       0
Bank Sta=4935.7,4944.5
Exp/Cntr=0.3,0.1

Type RM Length L Ch R = 1,27840,542,542,542
BEGIN DESCRIPTION:
Mapping XS 2fdc7b55
END DESCRIPTION:
XS GIS Cut Line= 3
      2110378.19     13412642.25      2109919.84     13411496.39
      2108509.18     13410554.21
#Sta/Elev= 30
  3094.7  322.54  3117.7  321.51  3171.6  317.59  3195.8  314.77  3249.6  310.38
  3279.3  309.34  3303.5  307.49  3333.1  306.55  3393.3  302.44  3465.1  299.58
  3501.0  299.01  3641.0  297.01  3739.7  297.05  3788.2  296.22  4140.9  294.99
  4635.3  294.73  4788.0  295.17  4947.2  294.88  4984.9  294.18  4985.7  293.38
  4992.9  293.38  4993.7  294.18  5034.8  295.37  5211.2  295.45  5303.4  295.26
  5457.8  294.99  5689.1  296.27  5898.5  296.19  6017.5  297.23  6025.2  297.40
#Mann=8,-1,0
  3094.7     0.1       0  4984.9    0.07       0  4993.7     0.1       0
  5034.8    0.05       0  5211.2     0.1       0  5303.4    0.05       0
  5898.5     0.1       0  6017.5    0.05       0
Bank Sta=4984.9,4993.7
Exp/Cntr=0.3,0.1

Type RM Length L Ch R = 1,27298,665,665,665
BEGIN DESCRIPTION:
Mapping XS dc312bb5
END DESCRIPTION:
XS GIS Cut Line= 4
      2110852.12     13412001.56      2110643.80     13411397.43
      2109154.22     13410345.35      2108389.26     13410543.09
#Sta/Elev= 30
  3215.9  300.10  3445.0  298.10  3550.7  298.03  3776.4  296.10  3815.2  296.32
  3920.3  295.21  4092.7  294.65  4235.5  293.55  4479.2  293.68  4574.1  294.33
  4773.5  293.48  4981.6  294.27  5012.8  293.16  5013.6  292.36  5020.8  292.36
  5021.6  293.16  5061.6  294.24  5362.0  293.86  5411.3  294.50  5492.5  294.71
  5555.3  295.56  5591.9  295.09  5740.1  295.98  6183.9  296.27  6235.5  297.49
  6289.1  297.87  6307.8  298.08  6335.1  297.35  6416.3  297.89  6468.7  297.46
#Mann=6,-1,0
  3215.9     0.1       0  5012.8    0.07       0  5021.6     0.1       0
  5411.3    0.05       0  5740.1     0.1       0  6289.1    0.05       0
Bank Sta=5012.8,5021.6
Exp/Cntr=0.3,0.1

Type RM Length L Ch R = 1,26633,502,502,502
BEGIN DESCRIPTION:
Mapping XS f94cfa06
END DESCRIPTION:
XS GIS Cut Line= 4
      2111065.67     13411913.01      2110841.72     13410881.81
      2109190.68     13409959.93      2108457.63     13410511.01
#Sta/Elev= 30
  3210.7  300.31  3311.0  299.53  3378.1  299.58  3505.4  298.17  3669.2  297.52
  3706.8  296.74  3925.0  295.46  3976.1  295.61  4468.3  293.28  4674.3  293.55
  4789.0  292.78  4820.6  291.89  4929.1  292.01  4968.1  291.12  4968.9  290.32
  4976.1  290.32  4976.9  291.12  5031.9  292.78  5069.6  292.56  5253.6  293.56
  5275.3  293.24  5313.0  293.77  5443.2  292.91  5583.7  292.93  6586.4  296.49
  6814.6  295.93  6907.2  296.46  6936.3  297.22  6980.9  296.88  7074.0  297.50
#Mann=4,-1,0
  3210.7     0.1       0  4968.1    0.07       0  4976.9     0.1       0
  6980.9    0.05       0
Bank Sta=4968.1,4976.9
Exp/Cntr=0.3,0.1

Type RM Length L Ch R = 1,26131,858,858,858
BEGIN DESCRIPTION:
Mapping XS c086f2cc
END DESCRIPTION:
XS GIS Cut Line= 4
      2111378.20     13411262.05      2110649.01     13410168.26
      2109242.76     13409663.06      2108451.11     13410449.49
#Sta/Elev= 30
  3271.8  297.73  3626.0  295.69  3662.0  295.02  4028.6  293.89  4181.7  292.55
  4302.0  294.20  4461.2  294.73  4726.3  293.96  4905.3  292.05  4973.2  291.90
  5022.9  292.89  5191.7  291.50  5192.6  290.70  5200.1  290.70  5201.0  291.50
  5437.2  292.37  5621.5  292.18  5764.5  292.96  5820.7  294.38  5912.9  294.76
  5961.4  295.59  6014.5  295.19  6186.5  296.54  6271.3  295.54  6370.3  296.41
  6412.8  295.71  6518.8  295.72  6787.5  296.49  7133.3  296.54  7196.5  296.84
#Mann=4,-1,0
  3271.8     0.1       0  5191.7    0.07       0  5201.0     0.1       0
  7133.3    0.05       0
Bank Sta=5191.7,5201
Exp/Cntr=0.3,0.1

Type RM Length L Ch R = 1,25273,66,66,66
BEGIN DESCRIPTION:
Mapping XS facd8223
END DESCRIPTION:
XS GIS Cut Line= 4
      2110946.71     13409990.65      2110056.96     13409404.71
      2109996.19     13409322.25      2108998.95     13409443.65
#Sta/Elev= 30
  3747.3  294.30  4170.5  293.90  4221.8  293.25  4360.0  293.38  4480.7  292.60
  4611.4  293.01  4769.9  292.29  4779.0  292.03  4806.0  289.66  4821.4  289.16
  4836.1  289.01  4842.3  289.52  4856.9  288.59  4918.2  287.97  4981.9  286.49
  4982.9  285.69  4990.8  285.69  4991.7  286.49  5062.2  288.19  5097.6  290.48
  5143.8  289.19  5148.9  289.87  5178.2  291.01  5289.0  291.94  5399.8  293.91
  5562.3  294.72  5601.3  295.41  5712.1  295.32  5742.3  296.16  5919.7  296.15
#Mann=3,-1,0
  3747.3     0.1       0  4981.9    0.07       0  4991.7     0.1       0
Bank Sta=4981.9,4991.7
Exp/Cntr=0.3,0.1

Type RM Length L Ch R = 1,25207,63,63,63
BEGIN DESCRIPTION:
Mapping XS ea15b129
END DESCRIPTION:
XS GIS Cut Line= 4
      2110925.00     13409873.46      2110143.76     13409369.99
      2110056.96     13409252.80      2108971.90     13409356.97
#Sta/Elev= 30
  3766.7  294.18  4135.5  293.65  4256.7  292.74  4547.2  293.14  4677.2  292.26
  4720.1  293.81  4734.7  293.43  4741.0  294.26  4764.0  294.39  4770.2  295.24
  4784.8  294.42  4791.1  295.17  4799.5  294.62  4805.7  295.50  4820.3  295.15
  4834.9  293.31  4924.3  294.55  5025.8  294.03  5044.8  294.85  5085.0  293.68
  5135.3  290.95  5170.5  290.28  5171.5  289.48  5179.4  289.48  5180.3  290.28
  5205.6  291.15  5476.8  294.57  5517.0  294.19  5748.1  295.72  5932.0  295.85
#Mann=3,-1,0
  3766.7     0.1       0  5170.5    0.07       0  5180.3     0.1       0
Bank Sta=5170.5,5180.3
Exp/Cntr=0.3,0.1

Type RM Length L Ch R = 1,25144,323,323,323
BEGIN DESCRIPTION:
Mapping XS 4d19aace
END DESCRIPTION:
XS GIS Cut Line= 4
      2111072.54     13409782.30      2110122.06     13409218.08
      2109766.16     13409200.72      2108978.12     13409252.68
#Sta/Elev= 30
  3657.9  294.50  3874.0  294.17  4033.8  293.07  4150.7  292.95  4252.0  292.32
  4310.5  292.59  4457.5  292.23  4485.9  292.59  4624.2  292.23  4661.2  291.71
  4756.7  291.18  4890.4  291.23  4980.5  290.48  5040.6  291.26  5090.7  291.11
  5110.7  290.00  5112.7  289.59  5113.7  288.79  5121.6  288.79  5122.5  289.59
  5170.8  291.06  5281.1  291.88  5321.1  292.70  5451.4  293.96  5501.5  293.87
  5521.6  294.33  5581.7  294.74  5711.8  294.71  5742.1  295.29  5909.3  295.89
#Mann=3,-1,0
  3657.9     0.1       0  5112.7    0.07       0  5122.5     0.1       0
Bank Sta=5112.7,5122.5
Exp/Cntr=0.3,0.1

Type RM Length L Ch R = 1,24821,806,806,806
BEGIN DESCRIPTION:
UNT 006 in La Jarita Watershed 20.0
END DESCRIPTION:
XS GIS Cut Line= 3
      2111143.82     13409334.94      2110025.00     13408925.00
      2108919.97     13408590.18
#Sta/Elev= 30
  3807.9  294.81  3883.5  295.04  3945.1  294.21  4050.5  293.88  4203.1  292.42
  4233.6  291.78  4319.8  291.35  4350.3  291.82  4406.0  291.16  4509.6  291.27
  4553.2  290.83  4648.0  291.00  4695.1  290.70  4756.1  290.90  4841.5  290.49
  4928.5  289.73  5016.4  289.75  5049.1  289.39  5050.1  288.59  5058.0  288.59
  5059.0  289.39  5208.4  290.48  5312.9  292.13  5431.8  293.43  5563.5  293.61
  5601.6  294.33  5639.7  294.15  5793.6  294.77  5856.3  294.55  6154.1  295.21
#Mann=5,-1,0
  3807.9     0.1       0  4841.5    0.05       0  5016.4     0.1       0
  5049.1    0.03       0  5059.0     0.1       0
Bank Sta=5049.1,5059
Exp/Cntr=0.3,0.1
