HEC-RAS study UNT 006 in La Jarita Watershed.prj: UNT 006 in La Jarita Watershed Base Level Engineering

--- UNT 006 in La Jarita Watershed.g01 (geometry) --- (continued)

Type RM Length L Ch R = 1,24015,321,321,321
BEGIN DESCRIPTION:
Mapping XS bf767d65
END DESCRIPTION:
XS GIS Cut Line= 3
      2111530.14     13409135.91      2109978.10     13408302.60
      2109155.17     13408026.55
#Sta/Elev= 30
  4167.9  295.14  4275.9  295.58  4349.6  294.67  4400.7  295.20  4431.6  294.59
  4468.8  294.64  4689.0  292.70  4710.9  292.15  4831.0  290.87  4946.3  288.67
  5039.6  288.67  5040.6  287.87  5048.6  287.87  5049.6  288.67  5170.4  289.48
  5219.9  288.99  5280.0  289.60  5323.9  289.16  5423.9  289.70  5436.9  289.64
  5559.3  290.33  5613.7  290.23  5672.0  291.32  5854.8  292.29  5893.0  292.16
  5928.4  292.82  6221.7  292.49  6531.9  293.50  6586.7  293.23  6797.5  293.66
#Mann=5,-1,0
  4167.9     0.1       0  5039.6    0.07       0  5049.6     0.1       0
  5423.9    0.05       0  5436.9     0.1       0
Bank Sta=5039.6,5049.6
Exp/Cntr=0.3,0.1

Type RM Length L Ch R = 1,23694,464,464,464
BEGIN DESCRIPTION:
Mapping XS 1de47f13
END DESCRIPTION:
XS GIS Cut Line= 3
      2111582.28     13408797.40      2111014.56     13408505.72
      2109630.53     13407839.72
#Sta/Elev= 30
  4253.4  294.40  4318.4  294.10  4351.5  294.37  4401.5  293.90  4440.2  294.15
  4475.2  293.40  4542.7  292.84  4623.3  291.60  4745.0  290.76  4795.2  289.64
  4811.8  289.76  4888.6  288.60  4986.1  287.88  4987.1  287.08  4995.1  287.08
  4996.1  287.88  5079.8  288.32  5138.2  289.19  5190.8  288.85  5251.3  289.49
  5296.6  289.32  5392.6  290.07  5477.6  289.90  5737.6  291.15  5856.7  291.17
  6060.0  292.02  6189.6  291.45  6263.6  292.41  6354.1  292.36  6427.6  292.74
#Mann=3,-1,0
  4253.4     0.1       0  4986.1    0.07       0  4996.1     0.1       0
Bank Sta=4986.1,4996.1
Exp/Cntr=0.3,0.1

Type RM Length L Ch R = 1,23230,465,465,465
BEGIN DESCRIPTION:
Mapping XS 67a76ac1
END DESCRIPTION:
XS GIS Cut Line= 4
      2111780.21     13408688.05      2111399.97     13408266.14
      2110879.14     13408031.76      2109962.50     13407703.65
#Sta/Elev= 30
  4100.7  294.26  4156.3  294.53  4276.7  293.77  4311.8  294.17  4340.2  293.67
  4354.4  294.08  4446.3  294.15  4495.7  293.03  4623.5  292.46  4802.8  289.45
  4849.1  288.28  4906.4  287.67  4952.7  287.94  4976.3  287.58  4977.3  286.78
  4985.4  286.78  4986.4  287.58  5022.2  288.24  5073.9  287.79  5189.5  288.47
  5278.0  290.16  5350.4  290.80  5482.8  290.81  5575.1  291.59  5723.6  291.16
  5796.5  292.05  5872.2  292.43  5984.6  292.18  6107.7  292.81  6213.4  292.83
#Mann=3,-1,0
  4100.7     0.1       0  4976.3    0.07       0  4986.4     0.1       0
Bank Sta=4976.3,4986.4
Exp/Cntr=0.3,0.1

Type RM Length L Ch R = 1,22765,56,56,56
BEGIN DESCRIPTION:
Mapping XS 15d17d3e
END DESCRIPTION:
XS GIS Cut Line= 6
      2111871.96     13408591.63      2111416.25     13407895.04
      2111140.64     13407669.35      2111069.03     13407678.03
      2111099.41     13407914.57      2110089.04     13407693.42
#Sta/Elev= 30
  3771.2  293.93  4429.4  291.62  4647.6  284.96  4711.3  286.88  4761.1  285.03
  4782.1  286.96  4811.1  284.97  4832.1  287.45  4847.0  284.99  4868.0  286.97
  4882.9  284.55  4914.7  283.94  4915.7  283.14  4924.8  283.94  4956.7  285.21
  4962.1  287.32  4970.8  284.87  5008.7  284.66  5034.4  288.81  5042.7  286.08
  5062.9  286.99  5068.2  285.17  5093.7  288.65  5099.0  286.74  5124.5  289.69
  5129.3  287.66  5240.0  289.69  5363.5  287.81  5609.2  291.46  6311.4  292.92
#Mann=3,-1,0
  3771.2     0.1       0  4914.7    0.07       0  4924.8     0.1       0
Bank Sta=4914.7,4924.8
Exp/Cntr=0.3,0.1

Type RM Length L Ch R = 1,22709,20,20,20
BEGIN DESCRIPTION:
Mapping XS 4d2c594d
END DESCRIPTION:
XS GIS Cut Line= 6
      2111903.23     13408582.11      2111417.12     13407835.58
      2111135.00     13407631.59      2111039.51     13407696.69
      2111078.57     13407839.92      2109748.09     13407597.23
#Sta/Elev= 30
  3697.7  294.22  3938.9  293.19  3974.9  294.34  4026.0  292.86  4320.5  292.08
  4380.0  290.59  4443.1  292.17  4479.7  290.96  4495.9  291.99  4501.6  290.77
  4517.8  292.65  4523.5  291.41  4555.7  292.76  4598.1  291.30  4668.6  293.21
  4740.6  290.38  4870.6  290.60  4948.7  292.21  4993.7  287.89  4994.7  287.09
  5003.8  287.89  5031.2  291.62  5075.1  289.54  5118.1  291.58  5152.6  290.59
  5187.2  291.14  5192.4  292.29  5258.3  287.96  5420.9  290.73  6576.6  293.85
#Mann=3,-1,0
  3697.7     0.1       0  4993.7    0.07       0  5003.8     0.1       0
Bank Sta=4993.7,5003.8
Exp/Cntr=0.3,0.1

Type RM Length L Ch R = 1,22689,549,549,549
BEGIN DESCRIPTION:
Mapping XS bc9f2a44
END DESCRIPTION:
XS GIS Cut Line= 6
      2111972.69     13408569.12      2111460.52     13407835.58
      2111208.78     13407631.59      2111035.17     13407605.55
      2111004.79     13407787.84      2109795.62     13407419.45
#Sta/Elev= 30
  3655.8  293.76  3951.4  292.70  4001.7  293.82  4109.4  291.73  4175.1  292.60
  4384.4  289.59  4426.2  290.30  4484.1  288.69  4519.4  290.48  4533.8  289.06
  4576.1  288.37  4675.4  288.84  4740.9  287.40  4741.9  286.60  4751.0  287.40
  4831.8  287.91  4861.1  289.03  4874.5  290.95  4877.7  290.95  4882.4  289.12
  4908.7  289.71  4914.0  288.25  4952.6  290.33  4993.0  287.69  5122.8  289.39
  5245.7  288.40  5411.4  291.36  5462.5  290.71  5661.1  291.96  6507.2  293.49
#Mann=3,-1,0
  3655.8     0.1       0  4740.9    0.07       0  4751.0     0.1       0
Bank Sta=4740.9,4751
Exp/Cntr=0.3,0.1

Type RM Length L Ch R = 1,22140,339,339,339
BEGIN DESCRIPTION:
Mapping XS e8c1464e
END DESCRIPTION:
XS GIS Cut Line= 4
      2112081.19     13408300.01      2111638.47     13407727.07
      2111447.50     13407336.45      2109793.88     13407345.13
#Sta/Elev= 30
  4050.5  292.76  4294.2  290.95  4350.3  292.20  4443.6  290.56  4593.0  289.62
  4642.8  288.27  4671.8  288.98  4707.2  288.05  4793.7  287.56  4877.0  287.92
  4968.8  286.63  4969.8  285.83  4977.9  285.83  4978.9  286.63  5001.9  286.72
  5018.9  287.54  5077.4  287.38  5207.4  289.39  5461.9  291.24  5621.9  290.87
  5731.9  289.42  5771.9  288.13  5811.9  289.47  5886.3  289.94  6001.9  289.40
  6111.9  289.97  6201.9  289.37  6331.9  291.24  6451.9  292.15  6863.0  293.34
#Mann=3,-1,0
  4050.5     0.1       0  4968.8    0.07       0  4978.9     0.1       0
Bank Sta=4968.8,4978.9
Exp/Cntr=0.3,0.1

Type RM Length L Ch R = 1,21801,459,459,459
BEGIN DESCRIPTION:
Mapping XS fb860d00
END DESCRIPTION:
XS GIS Cut Line= 4
      2112181.02     13408208.88      2112033.44     13407748.78
      2111773.02     13407297.39      2111243.51     13407167.18
#Sta/Elev= 30
  4153.8  292.13  4241.9  291.51  4288.6  291.52  4336.4  290.86  4390.2  290.91
  4409.9  290.47  4486.6  289.77  4513.5  290.49  4545.6  289.86  4609.5  289.41
  4636.4  288.76  4704.4  288.78  4806.4  287.28  4837.6  287.40  4895.3  286.10
  4967.2  286.52  4993.7  285.80  4994.7  285.00  5002.8  285.00  5003.8  285.80
  5033.9  286.56  5063.4  286.29  5137.8  286.59  5197.3  287.58  5273.7  287.66
  5351.6  288.61  5403.4  289.59  5460.7  289.76  5528.0  290.48  5703.4  290.88
#Mann=4,-1,0
  4153.8     0.1       0  4993.7    0.07       0  5003.8     0.1       0
  5460.7    0.05       0
Bank Sta=4993.7,5003.8
Exp/Cntr=0.3,0.1

Type RM Length L Ch R = 1,21342,568,568,568
BEGIN DESCRIPTION:
Mapping XS 14678552
END DESCRIPTION:
XS GIS Cut Line= 4
      2112284.31     13408294.16      2112174.93     13407325.38
      2111841.59     13406856.63      2111238.74     13407064.51
#Sta/Elev= 30
  3749.0  292.49  3790.4  292.11  3828.7  292.36  4054.9  290.81  4090.3  290.75
  4120.5  291.45  4160.8  290.32  4234.6  289.92  4311.7  288.65  4414.3  288.09
  4432.5  288.36  4492.9  287.64  4623.7  287.05  4678.9  287.41  4800.1  286.40
  4896.2  286.40  4954.1  285.44  4977.0  284.45  4978.0  283.65  4986.1  283.65
  4987.1  284.45  5004.5  285.02  5025.4  284.95  5305.1  289.79  5411.9  290.14
  5523.6  289.50  5623.4  289.75  5799.1  289.44  5866.8  290.39  5936.8  290.51
#Mann=4,-1,0
  3749.0     0.1       0  4800.1    0.05       0  4977.0    0.03       0
  4987.1    0.05       0
Bank Sta=4977,4987.1
Exp/Cntr=0.3,0.1

Type RM Length L Ch R = 1,20774,812,812,812
BEGIN DESCRIPTION:
UNT 006 in La Jarita Watershed 15.0
END DESCRIPTION:
XS GIS Cut Line= 4
      2112325.98     13408214.23      2112560.34     13407181.28
      2112282.57     13406469.48      2111129.04     13405983.78
#Sta/Elev= 30
  3497.6  291.93  3681.4  291.13  3732.7  291.67  4008.7  289.12  4358.2  288.02
  4422.2  286.76  4491.5  287.23  4530.7  286.72  4587.8  286.83  4636.8  286.08
  4696.5  286.24  4853.4  285.45  4943.7  284.69  4993.0  282.97  4994.0  282.17
  5002.1  282.17  5003.1  282.97  5022.6  284.44  5052.4  285.04  5320.6  286.62
  5752.2  283.89  5828.2  284.49  5881.8  283.93  5958.4  284.58  6040.4  284.15
  6208.0  285.53  6270.3  286.86  6381.6  287.94  6435.8  287.91  6572.5  289.02
#Mann=4,-1,0
  3497.6     0.1       0  4530.7    0.05       0  4993.0    0.03       0
  5003.1    0.05       0
Bank Sta=4993,5003.1
Exp/Cntr=0.3,0.1

Type RM Length L Ch R = 1,19962,305,305,305
BEGIN DESCRIPTION:
Mapping XS c68c00b8
END DESCRIPTION:
XS GIS Cut Line= 4
      2113360.68     13406745.49      2113183.61     13406443.44
      2112329.44     13406162.19      2111100.28     13405964.27
#Sta/Elev= 30
  4398.6  293.47  4476.8  293.33  4504.0  292.60  4711.3  290.66  4778.9  289.32
  4863.1  286.51  4936.8  285.03  4978.6  283.13  5010.4  283.43  5042.0  283.02
  5042.8  282.22  5052.1  282.22  5052.9  283.02  5157.9  284.03  5238.1  285.15
  5370.5  285.78  5402.2  285.53  5547.4  286.84  5726.6  284.33  5834.8  283.33
  6035.8  284.89  6199.5  284.10  6300.8  284.38  6381.8  284.78  6503.3  287.02
  6695.8  287.72  6736.3  288.32  6786.9  288.15  6859.9  288.80  6893.0  289.83
#Mann=4,-1,0
  4398.6     0.1       0  5042.0    0.07       0  5052.9     0.1       0
  5157.9    0.05       0
Bank Sta=5042,5052.9
Exp/Cntr=0.3,0.1

Type RM Length L Ch R = 1,19657,602,602,602
BEGIN DESCRIPTION:
Mapping XS 7d7ec603
END DESCRIPTION:
XS GIS Cut Line= 3
      2113834.63     13406479.88      2112683.61     13405901.77
      2111069.55     13405532.10
#Sta/Elev= 30
  4093.2  289.28  4224.0  288.83  4335.7  290.06  4408.3  290.12  4462.1  291.03
  4521.1  291.04  4596.3  290.50  4720.9  289.21  4787.9  287.14  4954.4  283.83
  4966.6  283.51  4983.3  281.74  4993.8  281.30  4994.6  280.50  5003.9  280.50
  5004.7  281.30  5005.6  282.12  5021.6  282.52  5228.9  285.03  5407.1  284.78
  5502.9  284.07  5554.2  284.29  5728.6  282.77  5879.6  284.95  6262.1  284.53
  6506.1  287.14  6640.0  287.33  6795.5  286.15  6939.2  286.36  7037.1  288.44
#Mann=6,-1,0
  4093.2     0.1       0  4521.1    0.05       0  4596.3     0.1       0
  4993.8    0.07       0  5004.7     0.1       0  5407.1    0.05       0
Bank Sta=4993.8,5004.7
Exp/Cntr=0.3,0.1

Type RM Length L Ch R = 1,19055,411,411,411
BEGIN DESCRIPTION:
UNT 006 in La Jarita Watershed 14.0
END DESCRIPTION:
XS GIS Cut Line= 3
      2114063.81     13406396.55      2112933.61     13405349.69
      2111100.32     13405250.73
#Sta/Elev= 30
  3708.7  291.28  3753.6  291.09  4098.2  287.90  4508.7  286.56  4706.6  283.95
  4926.0  282.21  4961.2  282.50  4977.3  281.87  4978.1  281.07  4987.4  281.07
  4988.2  281.87  5046.2  282.28  5124.5  284.10  5194.8  284.45  5230.5  285.26
  5287.9  285.15  5368.0  286.57  5418.1  286.14  5480.5  284.65  5613.9  282.38
  5778.6  284.86  5989.8  284.33  6319.4  284.47  6439.6  285.69  6619.8  285.39
  6649.9  285.91  6800.1  286.04  6850.2  287.10  7010.4  286.35  7085.2  287.19
#Mann=5,-1,0
  3708.7    0.08       0  3753.6     0.1       0  4977.3    0.07       0
  4988.2     0.1       0  5480.5    0.05       0
Bank Sta=4977.3,4988.2
Exp/Cntr=0.3,0.1

Type RM Length L Ch R = 1,18644,920,920,920
BEGIN DESCRIPTION:
UNT 006 in La Jarita Watershed 13.0
END DESCRIPTION:
XS GIS Cut Line= 3
      2114074.22     13406220.32      2113275.00     13405175.00
      2112854.96     13404389.39
#Sta/Elev= 30
  3670.7  291.58  3695.2  290.69  3732.3  290.94  3888.4  289.89  3959.1  288.51
  3988.1  288.79  4187.6  287.10  4223.0  286.41  4380.8  285.64  4407.9  285.07
  4445.2  285.22  4729.9  282.35  4950.2  282.08  4973.0  281.59  4989.2  280.64
  4990.0  279.84  4999.3  279.84  5000.1  280.64  5022.3  281.91  5044.2  282.17
  5229.6  282.31  5296.2  282.61  5340.1  283.55  5356.4  284.37  5400.3  284.45
  5451.5  285.67  5570.2  287.14  5652.3  286.60  5756.3  286.94  5877.4  286.24
#Mann=5,-1,0
  3670.7    0.08       0  3732.3     0.1       0  4989.2    0.07       0
  5000.1     0.1       0  5229.6    0.05       0
Bank Sta=4989.2,5000.1
Exp/Cntr=0.3,0.1

Type RM Length L Ch R = 1,17724,60,60,60
BEGIN DESCRIPTION:
Mapping XS 8864fb4c
END DESCRIPTION:
XS GIS Cut Line= 6
      2114267.81     13406442.57      2113795.83     13405560.35
      2113800.80     13404766.35      2113787.78     13404623.12
      2113692.29     13404497.26      2112924.74     13403921.93
#Sta/Elev= 30
  3126.0  292.01  3333.2  291.77  3408.8  290.65  3486.8  292.04  3546.9  290.55
  3605.9  290.18  3776.9  289.74  4122.1  285.95  4341.9  284.86  4601.9  281.45
  4721.9  281.36  4771.9  283.07  4803.4  282.00  4871.9  277.16  4923.7  276.19
  4927.7  275.02  4928.4  274.22  4937.9  274.22  4938.7  275.02  5002.2  276.25
  5038.6  279.12  5043.6  278.18  5072.8  281.14  5093.6  281.72  5172.6  281.92
  5351.2  284.68  5571.5  286.04  5819.4  285.49  5928.8  285.52  6181.6  286.11
#Mann=8,-1,0
  3126.0    0.05       0  3408.8    0.08       0  3605.9     0.1       0
  4927.7    0.07       0  4938.7     0.1       0  5351.2    0.05       0
  5819.4    0.08       0  5928.8    0.05       0
Bank Sta=4927.7,4938.7
Exp/Cntr=0.3,0.1

Type RM Length L Ch R = 1,17664,63,63,63
BEGIN DESCRIPTION:
Mapping XS d2a94903
END DESCRIPTION:
XS GIS Cut Line= 4
      2114330.32     13406470.36      2113873.49     13405553.65
      2113851.83     13404619.86      2113044.52     13403671.92
#Sta/Elev= 30
  3105.1  292.14  3435.1  291.67  3536.9  290.57  3613.9  291.91  3693.2  290.29
  3744.4  290.10  4328.0  285.65  4388.0  283.87  4458.1  284.16  4692.6  281.19
  4693.4  280.39  4702.9  280.39  4703.6  281.19  4718.1  281.58  4768.2  287.48
  4788.2  287.79  4858.2  287.04  5079.0  288.11  5093.3  287.84  5099.8  287.05
  5121.8  287.14  5171.2  281.83  5185.5  281.60  5376.5  284.61  5542.9  285.46
  5770.2  285.22  5903.3  285.32  5979.4  284.90  6085.9  285.89  6308.5  286.00
#Mann=8,-1,0
  3105.1    0.05       0  3536.9    0.08       0  3744.4     0.1       0
  4692.6    0.07       0  4703.6     0.1       0  5542.9    0.05       0
  5770.2    0.08       0  5903.3    0.05       0
Bank Sta=4692.6,4703.6
Exp/Cntr=0.3,0.1

Type RM Length L Ch R = 1,17601,107,107,107
BEGIN DESCRIPTION:
Mapping XS 0936ff5f
END DESCRIPTION:
XS GIS Cut Line= 5
      2114431.02     13406591.92      2113963.17     13405522.35
      2113926.66     13404874.86      2113909.30     13404545.00
      2113149.38     13403651.90
#Sta/Elev= 30
  2987.9  292.56  3508.4  291.59  3708.1  289.99  3811.3  291.36  3937.3  289.37
  4038.1  289.04  4222.8  286.53  4322.9  286.27  4763.6  281.21  4843.7  281.72
  4913.8  280.61  4929.7  279.32  4934.8  280.40  4988.5  278.21  4989.2  277.41
  4998.7  277.41  4999.5  278.21  5044.0  279.15  5084.1  281.09  5222.6  281.17
  5499.3  285.38  5649.9  285.03  5737.3  285.24  5870.4  285.17  5892.3  284.97
  5917.7  284.69  5967.1  285.73  6087.9  285.12  6264.7  286.30  6306.8  285.79
#Mann=9,-1,0
  2987.9    0.05       0  3708.1    0.08       0  3937.3     0.1       0
  4988.5    0.07       0  4999.5     0.1       0  5649.9    0.05       0
  5737.3    0.08       0  5870.4     0.1       0  5892.3    0.05       0
Bank Sta=4988.5,4999.5
Exp/Cntr=0.3,0.1

Type RM Length L Ch R = 1,17494,353,353,353
BEGIN DESCRIPTION:
Mapping XS d608e40b
END DESCRIPTION:
XS GIS Cut Line= 4
      2114514.33     13406581.45      2114026.55     13405439.08
      2114010.51     13404055.97      2113239.85     13403420.69
#Sta/Elev= 30
  2967.0  292.73  3636.0  290.54  3823.0  290.78  3898.1  289.54  4017.3  290.12
  4131.6  287.14  4204.3  287.26  4503.2  284.43  4543.3  284.71  4603.3  281.70
  4653.3  284.38  4693.3  282.82  4863.3  280.37  5003.3  279.06  5113.3  280.03
  5187.8  277.97  5188.5  277.17  5198.0  277.17  5198.8  277.97  5253.3  278.33
  5313.3  280.49  5393.3  279.84  5483.3  281.97  5601.6  283.25  5680.3  283.85
  5731.5  283.75  5788.9  284.80  6046.5  284.68  6298.3  284.84  6591.1  285.29
#Mann=9,-1,0
  2967.0    0.05       0  3898.1    0.08       0  4131.6     0.1       0
  5187.8    0.07       0  5198.8     0.1       0  5601.6    0.08       0
  5680.3    0.05       0  6046.5     0.1       0  6298.3    0.05       0
Bank Sta=5187.8,5198.8
Exp/Cntr=0.3,0.1

Type RM Length L Ch R = 1,17141,519,519,519
BEGIN DESCRIPTION:
UNT 006 in La Jarita Watershed 11.0
END DESCRIPTION:
XS GIS Cut Line= 4
      2114625.44     13406223.80      2114157.25     13405373.23
      2114193.67     13404031.67      2113312.56     13403321.57
#Sta/Elev= 30
  3063.7  291.35  3277.9  290.31  3474.0  290.34  3533.6  289.49  3908.6  289.30
  4006.1  288.40  4030.2  287.33  4501.2  283.63  4506.2  284.02  4693.1  282.40
  4773.1  282.30  4853.1  280.52  4907.5  280.16  4997.7  279.24  4998.4  278.44
  5008.0  278.44  5008.7  279.24  5023.2  279.81  5083.2  279.27  5263.3  279.37
  5401.2  280.13  5458.7  283.95  5479.5  283.89  5522.7  282.32  5533.2  282.56
  5636.3  283.95  5970.0  284.20  6286.6  284.61  6404.0  285.20  6508.3  284.74
#Mann=8,-1,0
  3063.7    0.05       0  4030.2    0.08       0  4907.5     0.1       0
  4997.7    0.07       0  5008.7     0.1       0  5533.2    0.05       0
  5970.0     0.1       0  6286.6    0.05       0
Bank Sta=4997.7,5008.7
Exp/Cntr=0.3,0.1

Type RM Length L Ch R = 1,16622,97,97,97
BEGIN DESCRIPTION:
Mapping XS 20421448
END DESCRIPTION:
XS GIS Cut Line= 4
      2114992.30     13404458.77      2114594.89     13403960.14
      2114221.63     13403972.29      2113507.88     13403228.69
#Sta/Elev= 30
  4174.8  286.73  4444.3  286.42  4560.2  286.35  4702.7  284.33  4773.2  282.03
  4872.3  279.74  4922.4  277.14  4976.9  276.79  4977.6  275.99  4987.2  275.99
  4988.0  276.79  5032.4  278.55  5106.8  278.88  5111.5  278.83  5116.5  279.68
  5132.5  279.29  5212.9  280.07  5245.2  280.55  5287.7  282.29  5294.6  283.12
  5322.9  283.94  5344.3  283.95  5365.4  283.03  5419.7  283.75  5471.7  284.57
  5563.5  283.46  5781.3  283.86  5909.9  284.18  6030.2  284.54  6216.6  283.63
#Mann=9,-1,0
  4174.8    0.05       0  4444.3     0.1       0  4976.9    0.07       0
  4988.0     0.1       0  5106.8    0.05       0  5212.9     0.1       0
  5419.7    0.05       0  5781.3     0.1       0  5909.9    0.05       0
Bank Sta=4976.9,4988
Exp/Cntr=0.3,0.1

Type RM Length L Ch R = 1,16525,123,123,123
BEGIN DESCRIPTION:
Mapping XS 774ccf1d
END DESCRIPTION:
XS GIS Cut Line= 4
      2115145.06     13404368.47      2114575.62     13403871.08
      2114245.76     13403875.42      2113603.43     13403172.33
#Sta/Elev= 30
  4061.3  286.50  4426.2  286.73  4524.8  286.41  4616.9  284.94  4729.9  282.31
  4786.8  279.97  4795.5  279.05  4796.3  278.25  4805.9  278.25  4806.6  279.05
  4807.7  279.70  4814.5  280.01  4858.0  280.88  5089.5  283.46  5118.0  283.39
  5145.2  282.40  5155.2  282.86  5169.4  280.94  5183.6  279.81  5205.4  280.37
  5254.5  281.27  5282.9  282.42  5289.7  283.24  5324.8  284.20  5360.6  283.84
  5381.5  282.95  5411.8  283.23  5742.9  283.40  5926.7  284.33  6099.6  283.76
#Mann=7,-1,0
  4061.3    0.05       0  4426.2     0.1       0  4795.5    0.07       0
  4806.6     0.1       0  5089.5    0.05       0  5205.4     0.1       0
  5411.8    0.05       0
Bank Sta=4795.5,4806.6
Exp/Cntr=0.3,0.1

Type RM Length L Ch R = 1,16402,668,668,668
BEGIN DESCRIPTION:
Mapping XS 40c89af2
END DESCRIPTION:
XS GIS Cut Line= 4
      2115183.26     13404205.28      2114713.64     13403799.03
      2114245.76     13403726.11      2113742.31     13403150.62
#Sta/Elev= 30
  4065.5  286.46  4213.2  286.64  4270.2  287.29  4405.5  286.47  4489.6  286.30
  4560.9  284.68  4581.7  284.90  4735.7  281.32  4766.0  280.37  4786.3  278.65
  4796.4  278.26  4836.9  279.43  4948.2  278.58  4993.3  277.68  4994.0  276.88
  5003.6  276.88  5004.4  277.68  5097.2  280.07  5164.0  280.34  5212.7  281.70
  5303.2  283.27  5338.3  284.38  5381.0  284.07  5387.7  283.35  5399.3  283.21
  5593.6  283.22  5679.0  282.78  5806.7  283.72  5833.1  283.80  5924.6  283.84
#Mann=9,-1,0
  4065.5    0.05       0  4405.5     0.1       0  4993.3    0.07       0
  5004.4     0.1       0  5097.2    0.05       0  5212.7     0.1       0
  5399.3    0.05       0  5806.7     0.1       0  5833.1    0.05       0
Bank Sta=4993.3,5004.4
Exp/Cntr=0.3,0.1

Type RM Length L Ch R = 1,15734,542,542,542
BEGIN DESCRIPTION:
Mapping XS fd2f4900
END DESCRIPTION:
XS GIS Cut Line= 3
      2115637.07     13404310.77      2114541.16     13403019.55
      2113911.83     13402748.29
#Sta/Elev= 30
  3522.2  285.73  3698.4  286.26  3840.1  285.99  3983.4  286.70  4187.2  286.47
  4308.0  285.91  4329.9  285.20  4365.1  285.63  4556.2  282.50  4599.1  281.10
  4818.8  276.85  4870.3  276.69  4871.1  275.89  4880.7  275.89  4881.4  276.69
  4882.8  276.90  4939.6  276.99  5046.1  278.63  5109.8  280.35  5268.3  282.21
  5498.2  280.22  5538.0  280.83  5619.4  280.95  5642.9  283.15  5658.1  283.35
  5671.9  283.40  5701.6  282.16  5728.8  282.64  5810.5  283.13  5901.1  282.13
#Mann=7,-1,0
  3522.2    0.05       0  3983.4     0.1       0  4870.3    0.03       0
  4881.4     0.1       0  4882.8    0.05       0  5498.2    0.08       0
  5728.8    0.05       0
Bank Sta=4870.3,4881.4
Exp/Cntr=0.3,0.1

Type RM Length L Ch R = 1,15192,501,501,501
BEGIN DESCRIPTION:
Mapping XS a9681255
END DESCRIPTION:
XS GIS Cut Line= 4
      2115205.31     13403708.16      2115109.00     13402915.80
      2114906.69     13402704.46      2114212.23     13402519.99
#Sta/Elev= 30
  3942.7  285.91  4234.2  280.68  4328.7  280.43  4401.6  278.82  4484.4  277.63
  4580.1  277.86  4786.6  280.12  4884.9  277.84  4970.6  276.36  4998.9  274.83
  5027.2  275.61  5045.6  272.79  5050.8  270.43  5066.2  268.21  5076.6  266.85
  5102.1  265.75  5102.8  264.95  5112.4  264.95  5113.2  265.75  5131.1  266.32
  5149.0  268.70  5180.1  275.63  5211.5  279.02  5246.5  279.96  5293.9  277.20
  5367.0  277.43  5531.5  281.21  5637.8  282.79  5716.6  282.39  5752.0  281.63
#Mann=8,-1,0
  3942.7     0.1       0  4401.6    0.05       0  4580.1    0.07       0
  4884.9    0.05       0  5102.1    0.03       0  5113.2    0.05       0
  5531.5     0.1       0  5716.6    0.08       0
Bank Sta=5102.1,5113.2
Exp/Cntr=0.3,0.1

Type RM Length L Ch R = 1,14691,528,528,528
BEGIN DESCRIPTION:
Mapping XS 24442cc5
END DESCRIPTION:
XS GIS Cut Line= 4
      2115583.78     13402762.70      2115385.87     13402442.57
      2114852.01     13402095.35      2114491.73     13402056.28
#Sta/Elev= 30
  4424.8  279.50  4503.3  278.73  4551.7  278.62  4597.9  277.93  4655.2  277.91
  4719.6  277.90  4756.2  277.38  4858.4  277.25  4946.6  275.88  4967.1  275.46
  5009.3  275.52  5076.2  275.00  5076.9  274.20  5086.6  274.20  5087.3  275.00
  5160.2  276.31  5211.4  276.63  5226.7  276.42  5247.8  276.96  5299.2  277.50
  5356.5  279.19  5413.8  279.98  5489.0  280.17  5575.6  279.62  5637.8  279.93
  5672.3  279.59  5686.5  279.97  5736.8  280.07  5768.9  280.52  5800.4  280.26
#Mann=7,-1,0
  4424.8     0.1       0  4655.2    0.05       0  4946.6    0.07       0
  5076.2    0.07       0  5087.3    0.07       0  5211.4     0.1       0
  5637.8    0.05       0
Bank Sta=5076.2,5087.3
Exp/Cntr=0.3,0.1

Type RM Length L Ch R = 1,14163,128,128,128
BEGIN DESCRIPTION:
UNT 006 in La Jarita Watershed 10.0
END DESCRIPTION:
XS GIS Cut Line= 4
      2115911.05     13403124.03      2115725.00     13402325.00
      2115452.36     13401996.55      2114684.46     13402027.64
#Sta/Elev= 30
  4211.8  278.69  4426.4  277.58  4488.0  278.11  4559.9  278.11  4631.8  277.46
  4652.3  276.78  4683.1  277.22  4816.6  277.50  4980.9  276.44  5053.7  276.90
  5088.8  279.14  5096.7  278.93  5103.2  278.14  5124.0  277.37  5167.0  277.10
  5259.4  278.11  5351.9  278.33  5488.6  277.58  5548.4  276.92  5586.5  276.14
  5666.5  275.49  5671.1  275.48  5671.8  274.68  5681.5  274.68  5682.2  275.48
  5863.5  278.29  5961.9  279.34  6096.9  281.04  6167.0  280.42  6227.6  280.53
#Mann=8,-1,0
  4211.8     0.1       0  5488.6    0.05       0  5548.4     0.1       0
  5666.5    0.07       0  5671.1    0.07       0  5682.2    0.07       0
  5863.5     0.1       0  5961.9    0.05       0
Bank Sta=5671.1,5682.2
Exp/Cntr=0.3,0.1

Type RM Length L Ch R = 1,14035,477,477,477
BEGIN DESCRIPTION:
Mapping XS 8235f0a1
END DESCRIPTION:
XS GIS Cut Line= 4
      2116019.54     13403197.76      2115867.64     13402407.85
      2115724.41     13401552.81      2115746.04     13401098.56
#Sta/Elev= 30
  4146.3  278.76  4201.0  278.95  4403.6  277.31  4460.6  277.15  4607.4  277.56
  4709.2  277.21  4749.9  277.50  4841.6  276.89  4949.6  276.57  4993.0  276.73
  5024.5  276.45  5180.1  277.41  5207.1  277.13  5288.2  277.19  5338.9  277.79
  5521.4  276.66  5592.3  276.54  5622.8  276.86  5653.2  276.33  5660.0  275.89
  5660.7  275.09  5670.4  275.09  5671.1  275.89  5721.2  276.58  5865.5  276.79
  5995.6  277.81  6045.7  277.72  6095.8  278.43  6135.8  278.28  6272.4  280.55
#Mann=3,-1,0
  4146.3     0.1       0  5660.0    0.07       0  5671.1     0.1       0
Bank Sta=5660,5671.1
Exp/Cntr=0.3,0.1

Type RM Length L Ch R = 1,13558,375,375,375
BEGIN DESCRIPTION:
UNT 006 in La Jarita Watershed 9.0
END DESCRIPTION:
XS GIS Cut Line= 3
      2116084.65     13403301.99      2116175.00     13402225.00
      2116227.88     13401170.90
#Sta/Elev= 30
  3788.6  279.14  3825.7  278.39  3865.9  278.99  3916.0  278.59  3966.2  278.71
  4146.8  276.95  4247.2  276.77  4277.3  276.38  4357.6  277.01  4588.4  277.69
  4668.7  276.75  4691.9  276.81  4759.0  275.46  4839.3  276.01  4966.8  274.45
  4999.5  274.41  5039.6  274.95  5114.1  274.23  5114.8  273.43  5124.5  273.43
  5125.2  274.23  5149.7  274.72  5199.8  274.96  5229.8  275.95  5279.9  276.00
  5410.1  277.66  5690.4  277.37  5800.5  278.74  5840.6  279.68  5924.8  280.47
#Mann=3,-1,0
  3788.6     0.1       0  5114.1    0.07       0  5125.2     0.1       0
Bank Sta=5114.1,5125.2
Exp/Cntr=0.3,0.1

Type RM Length L Ch R = 1,13183,698,698,698
BEGIN DESCRIPTION:
Mapping XS 1882970e
END DESCRIPTION:
XS GIS Cut Line= 4
      2116132.40     13403267.21      2116527.36     13402611.84
      2116505.66     13401696.04      2116427.79     13401168.29
#Sta/Elev= 30
  3793.5  278.18  3884.7  278.63  3921.6  278.22  3964.3  278.34  3994.6  277.88
  4038.1  277.97  4075.0  277.33  4139.0  277.10  4197.3  276.36  4298.3  274.48
  4372.0  273.66  4424.5  273.70  4525.4  272.51  4659.9  272.33  4660.7  271.53
  4670.4  271.53  4671.1  272.33  4845.6  273.96  4935.6  272.86  5035.7  272.72
  5085.7  273.51  5225.7  276.77  5296.1  277.75  5506.1  277.02  5688.1  276.93
  5768.9  277.47  5829.6  278.34  5855.4  279.21  5920.0  280.46  6008.2  281.04
#Mann=3,-1,0
  3793.5     0.1       0  4659.9    0.07       0  4671.1     0.1       0
Bank Sta=4659.9,4671.1
Exp/Cntr=0.3,0.1

Type RM Length L Ch R = 1,12485,352,352,352
BEGIN DESCRIPTION:
UNT 006 in La Jarita Watershed 8.0
END DESCRIPTION:
XS GIS Cut Line= 3
      2117392.29     13402469.22      2116875.00     13401925.00
      2116566.12     13401129.51
#Sta/Elev= 30
  4260.0  276.56  4285.1  276.51  4367.1  276.18  4416.8  275.31  4507.1  274.82
  4614.7  274.22  4734.9  272.37  4883.6  272.25  4954.4  271.67  4982.7  270.27
  4984.0  269.84  4984.7  269.04  4994.5  269.04  4995.2  269.84  4996.9  270.48
  5003.8  270.79  5007.4  271.44  5025.8  272.20  5074.9  272.74  5194.5  274.97
  5243.6  274.92  5273.5  275.56  5298.0  275.36  5397.0  276.18  5466.7  276.17
  5491.3  276.71  5536.5  276.90  5697.4  280.38  5804.7  281.09  5864.2  280.83
#Mann=5,-1,0
  4260.0     0.1       0  4285.1    0.05       0  4507.1     0.1       0
  4984.0    0.07       0  4995.2     0.1       0
Bank Sta=4984,4995.2
Exp/Cntr=0.3,0.1

Type RM Length L Ch R = 1,12133,616,616,616
BEGIN DESCRIPTION:
UNT 006 in La Jarita Watershed 7.0
END DESCRIPTION:
XS GIS Cut Line= 3
      2117628.38     13402399.75      2117183.08     13401826.07
      2116864.52     13401122.02
#Sta/Elev= 30
  4129.4  276.98  4163.2  276.92  4206.7  276.32  4262.8  275.99  4306.2  275.32
  4335.2  274.48  4413.9  273.64  4441.1  273.78  4548.8  273.15  4584.1  272.63
  4669.2  272.52  4698.2  272.20  4768.7  272.12  4833.0  272.43  4949.5  270.83
  4950.2  270.03  4960.1  270.03  4960.7  270.83  4977.5  271.08  5004.7  270.91
  5035.4  271.43  5087.3  273.30  5119.0  273.98  5225.7  275.94  5277.4  276.34
  5369.9  277.89  5438.5  278.32  5548.3  279.71  5587.8  279.77  5628.4  279.96
#Mann=6,-1,0
  4129.4    0.05       0  4949.5    0.03       0  4960.7    0.05       0
  5004.7     0.1       0  5119.0    0.05       0  5587.8     0.1       0
Bank Sta=4949.5,4960.7
Exp/Cntr=0.3,0.1

Type RM Length L Ch R = 1,11517,459,459,459
BEGIN DESCRIPTION:
Mapping XS 65979ebe
END DESCRIPTION:
XS GIS Cut Line= 4
      2118132.73     13402046.47      2117851.49     13401950.12
      2117523.37     13401588.14      2116893.12     13401082.91
#Sta/Elev= 30
  4390.9  279.09  4407.6  279.22  4483.6  278.49  4515.3  278.82  4569.3  278.24
  4642.2  278.50  4724.5  277.75  4758.4  276.97  4823.9  275.39  4901.6  272.88
  4965.1  270.44  4987.8  269.01  4988.5  268.21  4998.4  268.21  4999.1  269.01
  5050.3  270.83  5113.8  272.61  5199.8  273.84  5270.2  275.25  5303.9  274.96
  5348.7  275.14  5511.9  274.88  5575.9  275.77  5625.5  275.75  5725.8  277.36
  5789.8  277.90  5853.9  278.92  5896.0  278.91  5939.2  279.40  5984.5  279.48
#Mann=5,-1,0
  4390.9    0.05       0  4758.4     0.1       0  4987.8    0.07       0
  4999.1     0.1       0  5303.9    0.05       0
Bank Sta=4987.8,4999.1
Exp/Cntr=0.3,0.1

Type RM Length L Ch R = 1,11058,377,377,377
BEGIN DESCRIPTION:
UNT 006 in La Jarita Watershed 6.0
END DESCRIPTION:
XS GIS Cut Line= 3
      2118239.51     13402094.21      2118025.00     13401475.00
      2117088.34     13400963.15
#Sta/Elev= 30
  4308.9  280.47  4580.1  276.83  4673.6  274.53  4678.9  275.07  4742.0  274.64
  4761.7  273.89  4879.6  271.51  4900.7  270.72  4948.6  270.07  4981.3  268.39
  4981.4  268.39  4982.1  267.59  4992.0  267.59  4992.7  268.39  4993.9  268.42
  5009.8  269.01  5037.7  270.84  5053.9  271.03  5081.4  272.28  5097.5  272.58
  5103.2  273.06  5141.2  273.38  5184.8  274.35  5310.0  275.23  5375.5  274.89
  5413.5  275.27  5761.6  274.90  5892.6  276.64  5989.8  278.94  6031.6  279.55
#Mann=5,-1,0
  4308.9    0.05       0  4981.3     0.1       0  4981.4    0.03       0
  4992.7     0.1       0  4993.9    0.05       0
Bank Sta=4981.4,4992.7
Exp/Cntr=0.3,0.1

Type RM Length L Ch R = 1,10681,305,305,305
BEGIN DESCRIPTION:
Mapping XS d261f633
END DESCRIPTION:
XS GIS Cut Line= 3
      2118346.28     13402116.76      2118372.32     13401332.93
      2117128.76     13400950.50
#Sta/Elev= 30
  4317.4  278.96  4389.2  278.72  4489.3  276.89  4619.3  276.14  4666.5  275.41
  4765.1  274.59  4929.5  270.25  4979.5  269.49  5003.9  268.59  5004.6  267.79
  5014.5  267.79  5015.2  268.59  5049.6  270.35  5061.0  270.47  5098.1  271.79
  5140.6  272.15  5145.8  272.61  5172.1  272.58  5183.7  273.13  5243.9  273.73
  5249.1  274.14  5276.6  274.11  5287.2  274.56  5328.1  274.19  5412.7  274.59
  5475.5  275.67  5559.2  274.86  6196.2  274.94  6249.7  275.46  6402.7  279.19
#Mann=7,-1,0
  4317.4    0.05       0  4666.5     0.1       0  4765.1    0.05       0
  5003.9   0.033       0  5015.2    0.05       0  5061.0     0.1       0
  5328.1    0.05       0
Bank Sta=5003.9,5015.2
Exp/Cntr=0.3,0.1

Type RM Length L Ch R = 1,10376,325,325,325
BEGIN DESCRIPTION:
Mapping XS 29172e1c
END DESCRIPTION:
XS GIS Cut Line= 3
      2118694.37     13402042.10      2118670.07     13401312.97
      2118444.40     13401063.00
#Sta/Elev= 30
  4392.1  276.86  4508.3  275.77  4539.3  275.39  4569.3  275.58  4619.3  275.34
  4669.4  274.62  4719.4  274.62  4749.5  274.04  4824.0  272.63  4859.5  271.51
  4929.5  269.91  4949.5  269.88  4979.5  269.13  4993.9  268.21  4994.6  267.41
  5004.5  267.41  5005.2  268.21  5009.5  268.68  5019.5  269.00  5051.7  269.39
  5118.1  271.82  5140.1  272.36  5173.0  273.26  5194.7  274.38  5229.8  274.88
  5258.2  274.71  5286.6  275.03  5329.2  276.18  5406.9  275.50  5458.4  275.81
#Mann=7,-1,0
  4392.1    0.05       0  4508.3     0.1       0  4749.5    0.05       0
  4993.9   0.033       0  5005.2    0.05       0  5051.7     0.1       0
  5140.1    0.05       0
Bank Sta=4993.9,5005.2
Exp/Cntr=0.3,0.1

Type RM Length L Ch R = 1,10051,286,286,286
BEGIN DESCRIPTION:
Mapping XS 0792c044
END DESCRIPTION:
XS GIS Cut Line= 3
      2118944.37     13402101.16      2119017.29     13401191.44
      2118732.52     13401076.84
#Sta/Elev= 30
  4352.9  276.52  4379.1  276.06  4409.2  276.08  4449.4  275.37  4534.0  274.92
  4612.4  274.53  4640.0  274.05  4669.4  274.22  4710.2  273.93  4767.2  272.94
  4802.2  271.98  4867.2  271.02  4940.9  269.33  4985.5  267.62  4986.2  266.82
  4996.1  266.82  4996.8  267.62  5014.5  267.72  5021.2  267.80  5047.7  269.57
  5131.6  273.06  5231.9  275.56  5271.4  274.90  5319.7  274.78  5346.8  275.12
  5352.6  275.28  5432.6  276.00  5499.0  275.73  5538.2  275.75  5572.5  275.51
#Mann=12,-1,0
  4352.9    0.05       0  4534.0     0.1       0  4612.4    0.05       0
  4767.2     0.1       0  4867.2    0.05       0  4985.5    0.03       0
  4996.8    0.05       0  5014.5     0.1       0  5346.8    0.05       0
  5352.6     0.1       0  5499.0    0.05       0  5538.2     0.1       0
Bank Sta=4985.5,4996.8
Exp/Cntr=0.3,0.1

Type RM Length L Ch R = 1,9765,311,311,311
BEGIN DESCRIPTION:
Mapping XS f4254a7b
END DESCRIPTION:
XS GIS Cut Line= 3
      2119249.93     13402278.26      2119274.23     13401358.11
      2119062.41     13401201.85
#Sta/Elev= 30
  4259.2  276.60  4492.5  275.80  4639.1  274.67  4692.6  274.50  4772.6  272.15
  4812.7  271.43  4842.7  270.39  4902.7  268.80  4972.7  267.66  4992.7  267.61
  4997.1  267.38  4997.8  266.58  5007.7  266.58  5008.4  267.38  5032.7  269.13
  5072.7  270.74  5102.8  272.42  5142.8  273.94  5178.7  275.02  5189.1  274.81
  5195.4  275.01  5210.0  274.96  5230.8  275.41  5260.1  275.35  5281.0  275.56
  5310.2  275.24  5366.2  275.28  5381.2  275.14  5410.5  275.42  5442.9  275.17
#Mann=4,-1,0
  4259.2    0.05       0  4997.1    0.03       0  5008.4    0.05       0
  5366.2     0.1       0
Bank Sta=4997.1,5008.4
Exp/Cntr=0.3,0.1

Type RM Length L Ch R = 1,9454,335,335,335
BEGIN DESCRIPTION:
Mapping XS ea9b030c
END DESCRIPTION:
XS GIS Cut Line= 3
      2119465.21     13402323.34      2119600.62     13401354.64
      2119358.82     13401251.01
#Sta/Elev= 30
  4315.4  276.80  4475.3  276.06  4563.9  276.25  4596.4  275.95  4640.4  275.91
  4667.1  275.26  4747.9  274.31  4783.3  272.41  4788.4  272.49  4798.4  272.13
  4854.8  269.67  4859.8  269.68  4899.4  268.46  4926.2  267.83  5004.8  267.31
  5005.4  266.51  5015.4  266.51  5016.1  267.31  5140.6  273.17  5145.7  273.18
  5222.5  276.04  5232.6  276.24  5288.6  276.65  5293.5  276.46  5305.2  276.69
  5334.2  276.19  5386.8  275.96  5462.9  275.92  5504.6  276.13  5556.6  275.97
#Mann=3,-1,0
  4315.4    0.05       0  5004.8    0.03       0  5016.1    0.05       0
Bank Sta=5004.8,5016.1
Exp/Cntr=0.3,0.1

Type RM Length L Ch R = 1,9119,197,197,197
BEGIN DESCRIPTION:
Mapping XS 6e5ca436
END DESCRIPTION:
XS GIS Cut Line= 3
      2119763.81     13402406.76      2119895.76     13401552.55
      2119795.05     13401365.02
#Sta/Elev= 30
  4381.8  276.06  4488.8  276.30  4545.5  277.06  4688.3  276.33  4788.3  274.18
  4849.0  272.00  4882.7  271.38  4940.1  268.80  4945.8  268.27  4950.8  268.29
  4995.2  266.49  4995.8  265.69  5005.8  265.69  5006.5  266.49  5061.5  267.53
  5077.0  268.32  5112.1  269.02  5140.2  270.34  5145.2  270.11  5208.3  273.49
  5213.4  273.39  5253.7  274.98  5259.4  274.80  5275.6  275.64  5281.3  275.51
  5297.5  276.07  5325.1  276.09  5363.3  276.98  5407.1  276.83  5459.0  277.20
#Mann=3,-1,0
  4381.8    0.05       0  4995.2    0.03       0  5006.5    0.05       0
Bank Sta=4995.2,5006.5
Exp/Cntr=0.3,0.1

Type RM Length L Ch R = 1,8922,353,353,353
BEGIN DESCRIPTION:
Mapping XS 37557d17
END DESCRIPTION:
XS GIS Cut Line= 2
      2119986.04     13402472.72      2120086.69     13401469.66
#Sta/Elev= 30
  4360.1  277.46  4448.3  277.28  4508.6  277.50  4528.7  277.21  4597.0  277.06
  4602.1  277.21  4739.7  275.24  4769.9  274.47  4870.4  270.94  4898.0  270.90
  4910.6  270.56  4970.9  266.85  4985.3  266.26  4986.0  265.46  4996.0  265.46
  4996.6  266.26  4998.4  266.45  5003.4  266.30  5041.2  267.00  5071.4  267.99
  5091.5  268.83  5098.7  269.39  5103.7  269.45  5121.6  270.65  5141.7  271.69
  5192.0  273.42  5222.1  274.80  5299.3  277.00  5342.7  277.50  5368.2  277.52
#Mann=3,-1,0
  4360.1    0.05       0  4985.3    0.03       0  4996.6    0.05       0
Bank Sta=4985.3,4996.6
Exp/Cntr=0.3,0.1

Type RM Length L Ch R = 1,8569,35,35,35
BEGIN DESCRIPTION:
Mapping XS 15c3dc20
END DESCRIPTION:
XS GIS Cut Line= 4
      2120239.51     13402486.58      2120406.18     13402073.39
      2120399.23     13401764.36      2120211.74     13401562.98
#Sta/Elev= 30
  4325.3  276.21  4490.6  273.85  4699.9  271.78  4779.2  270.25  4799.2  269.17
  4819.2  268.65  4859.3  269.69  4916.2  268.94  4989.3  268.27  5009.3  268.58
  5039.3  269.71  5044.4  267.39  5045.1  266.59  5055.1  266.59  5055.7  267.39
  5072.0  268.48  5082.9  268.77  5089.7  269.52  5096.5  268.24  5103.9  269.27
  5110.7  268.27  5118.0  269.90  5124.9  269.53  5132.2  270.90  5139.0  270.73
  5146.4  271.85  5167.4  272.07  5209.9  273.56  5280.7  275.33  5355.1  276.21
#Mann=5,-1,0
  4325.3    0.05       0  4916.2     0.1       0  5044.4    0.07       0
  5055.7     0.1       0  5072.0    0.05       0
Bank Sta=5044.4,5055.7
Exp/Cntr=0.3,0.1

Type RM Length L Ch R = 1,8534,58,58,58
BEGIN DESCRIPTION:
Mapping XS 3fd5c249
END DESCRIPTION:
XS GIS Cut Line= 4
      2120246.45     13402510.90      2120440.90     13402181.02
      2120433.96     13401726.16      2120211.76     13401535.22
#Sta/Elev= 30
  4279.1  276.06  4310.4  275.33  4363.1  274.82  4427.5  273.65  4480.2  273.51
  4603.2  272.27  4698.0  271.01  4728.1  270.91  4778.1  269.71  4802.4  268.50
  4803.1  267.70  4813.1  267.70  4813.7  268.50  4828.1  269.54  4848.1  271.76
  4858.1  272.46  4878.1  273.30  4899.6  273.47  4948.1  273.90  4978.1  273.63
  4998.1  274.01  5064.4  274.37  5078.1  274.35  5115.0  272.74  5138.5  272.83
  5159.4  272.56  5202.2  272.98  5265.8  274.67  5329.5  275.93  5409.9  276.88
#Mann=5,-1,0
  4279.1    0.05       0  4802.4    0.07       0  4813.7    0.05       0
  4899.6     0.1       0  5064.4    0.05       0
Bank Sta=4802.4,4813.7
Exp/Cntr=0.3,0.1

Type RM Length L Ch R = 1,8476,284,284,284
BEGIN DESCRIPTION:
Mapping XS 70092964
END DESCRIPTION:
XS GIS Cut Line= 4
      2120267.32     13402528.21      2120510.34     13402229.64
      2120489.51     13401740.05      2120213.09     13401518.92
#Sta/Elev= 30
  4226.1  275.59  4262.3  274.58  4276.6  274.81  4340.5  274.23  4375.7  273.35
  4447.6  272.62  4553.1  272.32  4610.6  271.35  4635.7  271.48  4715.8  270.25
  4765.9  269.06  4795.9  267.58  4835.9  268.40  4869.7  268.20  4990.4  266.38
  4991.1  265.58  5001.1  265.58  5001.7  266.38  5016.1  266.96  5052.2  269.38
  5085.4  271.88  5090.4  272.65  5115.2  273.41  5129.7  272.88  5136.1  272.26
  5193.7  272.53  5214.5  273.30  5243.3  273.55  5342.6  275.86  5455.1  277.00
#Mann=5,-1,0
  4226.1    0.05       0  4869.7     0.1       0  4990.4    0.07       0
  5001.7     0.1       0  5052.2    0.05       0
Bank Sta=4990.4,5001.7
Exp/Cntr=0.3,0.1

Type RM Length L Ch R = 1,8192,133,133,133
BEGIN DESCRIPTION:
Mapping XS d1e9bf87
END DESCRIPTION:
XS GIS Cut Line= 3
      2121319.35     13401937.97      2120999.93     13401951.86
      2120246.47     13401524.78
#Sta/Elev= 30
  4404.1  276.57  4447.2  276.53  4468.5  276.10  4668.7  269.35  4679.5  269.21
  4855.9  269.57  4923.9  268.61  4952.1  267.34  4968.0  265.94  4982.4  265.51
  4995.4  264.61  4999.2  264.06  4999.7  263.26  5011.1  263.26  5011.6  264.06
  5017.1  264.63  5027.2  264.98  5039.8  266.27  5089.3  267.55  5120.3  268.21
  5194.5  268.08  5304.2  271.88  5340.2  273.46  5377.7  274.37  5415.3  274.83
  5421.0  275.15  5436.9  275.12  5458.5  275.88  5474.4  275.79  5589.9  276.95
#Mann=7,-1,0
  4404.1    0.05       0  4668.7     0.1       0  4679.5    0.05       0
  4923.9     0.1       0  4999.2    0.07       0  5011.6     0.1       0
  5089.3    0.05       0
Bank Sta=4999.2,5011.6
Exp/Cntr=0.3,0.1

Type RM Length L Ch R = 1,8059,286,286,286
BEGIN DESCRIPTION:
Mapping XS 6013566f
END DESCRIPTION:
XS GIS Cut Line= 3
      2121510.36     13401830.33      2121097.15     13401809.50
      2120219.34     13401493.76
#Sta/Elev= 30
  4319.5  275.63  4455.0  277.48  4535.1  277.42  4585.2  276.23  4635.3  274.36
  4675.3  273.25  4721.8  271.07  4726.8  271.08  4731.8  270.66  4756.4  269.98
  4787.1  269.33  4853.8  269.08  4958.7  267.44  4984.4  264.27  4984.9  263.47
  4996.3  263.47  4996.8  264.27  5002.1  265.01  5011.8  265.79  5033.1  266.66
  5052.9  266.77  5083.6  267.54  5150.3  267.72  5170.4  268.14  5201.1  268.13
  5237.2  268.70  5380.1  273.85  5447.5  275.71  5497.7  276.35  5666.1  276.95
#Mann=3,-1,0
  4319.5    0.05       0  4984.4    0.03       0  4996.8    0.05       0
Bank Sta=4984.4,4996.8
Exp/Cntr=0.3,0.1

Type RM Length L Ch R = 1,7773,339,339,339
BEGIN DESCRIPTION:
UNT 006 in La Jarita Watershed 5.0
END DESCRIPTION:
XS GIS Cut Line= 3
      2121473.91     13401268.67      2121249.93     13401471.82
      2120145.83     13401450.00
#Sta/Elev= 30
  4288.4  276.33  4348.8  276.90  4440.7  276.58  4462.3  276.05  4561.0  274.84
  4645.7  272.59  4681.9  271.09  4805.8  267.66  4885.8  266.34  4945.8  266.81
  4965.8  266.64  4975.8  266.10  4985.8  264.95  4995.8  263.69  4999.6  262.51
  5000.1  261.71  5011.5  261.71  5012.0  262.51  5025.8  263.73  5035.8  265.28
  5055.8  266.55  5085.8  266.75  5235.8  270.98  5275.9  271.55  5335.9  273.25
  5405.9  274.76  5495.9  275.97  5555.9  275.86  5595.9  276.41  5695.1  276.87
#Mann=3,-1,0
  4288.4    0.05       0  4999.6    0.03       0  5012.0    0.05       0
Bank Sta=4999.6,5012
Exp/Cntr=0.3,0.1

Type RM Length L Ch R = 1,7434,261,261,261
BEGIN DESCRIPTION:
Mapping XS d0667e96
END DESCRIPTION:
XS GIS Cut Line= 3
      2121427.06     13401096.82      2120619.72     13401195.78
      2120079.00     13401419.35
#Sta/Elev= 30
  4429.5  276.69  4512.2  276.07  4643.1  273.55  4764.0  269.11  4786.8  268.61
  4824.5  267.04  4915.2  265.94  4955.5  263.98  4975.6  264.28  4989.6  263.19
  4990.1  262.39  5001.5  262.39  5002.0  263.19  5005.8  264.39  5031.0  265.88
  5056.2  266.11  5112.4  267.74  5146.9  268.24  5193.8  269.39  5237.6  269.54
  5323.7  269.03  5407.9  269.64  5466.6  270.69  5485.1  270.69  5519.8  271.71
  5567.6  272.23  5620.8  273.64  5644.7  273.89  5756.6  276.24  5828.0  277.02
#Mann=3,-1,0
  4429.5    0.05       0  4989.6    0.03       0  5002.0    0.05       0
Bank Sta=4989.6,5002
Exp/Cntr=0.3,0.1

Type RM Length L Ch R = 1,7173,584,584,584
BEGIN DESCRIPTION:
Mapping XS 91b36e83
END DESCRIPTION:
XS GIS Cut Line= 4
      2121562.41     13400565.58      2121119.72     13400846.82
      2120432.22     13401044.74      2120104.07     13401367.68
#Sta/Elev= 30
  4211.6  275.94  4280.7  275.36  4478.0  271.45  4623.2  271.06  4723.6  269.90
  4813.8  268.29  4892.0  265.77  4930.9  265.98  4959.4  263.88  4980.3  264.60
  4990.7  264.23  4997.3  263.25  4997.8  262.45  5009.2  262.45  5009.7  263.25
  5031.9  265.28  5042.8  265.54  5136.4  265.99  5261.3  268.33  5293.7  268.42
  5361.1  267.17  5394.8  267.10  5456.8  267.33  5499.2  268.15  5598.2  267.88
  5626.5  268.44  5661.8  269.93  5739.7  271.33  5859.8  275.14  5911.9  276.11
#Mann=3,-1,0
  4211.6    0.05       0  4997.3    0.03       0  5009.7    0.05       0
Bank Sta=4997.3,5009.7
Exp/Cntr=0.3,0.1

Type RM Length L Ch R = 1,6589,508,508,508
BEGIN DESCRIPTION:
Mapping XS 94a720b1
END DESCRIPTION:
XS GIS Cut Line= 5
      2121562.46     13400539.53      2120968.68     13400607.24
      2120671.80     13400643.70      2120296.80     13401081.20
      2119999.93     13401378.07
#Sta/Elev= 30
  3812.4  276.01  3905.1  274.42  4079.0  270.06  4173.4  269.40  4293.0  267.25
  4435.8  266.34  4512.1  267.99  4593.4  268.31  4743.2  267.54  4776.2  266.79
  4835.4  266.15  4863.9  265.13  4962.7  264.55  5005.5  262.49  5013.6  261.46
  5014.1  260.66  5025.5  260.66  5026.0  261.46  5026.9  262.28  5034.1  264.02
  5046.5  263.96  5119.1  263.94  5189.9  266.48  5218.5  268.08  5267.8  267.66
  5338.8  268.14  5388.3  270.28  5494.4  272.29  5607.5  275.39  5705.2  276.91
#Mann=5,-1,0
  3812.4    0.05       0  4776.2     0.1       0  5013.6    0.07       0
  5026.0     0.1       0  5046.5    0.05       0
Bank Sta=5013.6,5026
Exp/Cntr=0.3,0.1

Type RM Length L Ch R = 1,6081,196,196,196
BEGIN DESCRIPTION:
Mapping XS 78c73fcb
END DESCRIPTION:
XS GIS Cut Line= 2
      2120701.33     13400475.29      2119534.69     13400885.00
#Sta/Elev= 30
  4540.5  269.00  4610.3  269.05  4653.2  268.18  4813.2  266.74  4920.2  265.60
  4939.4  264.30  4945.9  262.24  4960.6  261.11  4975.9  260.92  4976.4  260.12
  4987.8  260.12  4988.3  260.92  5002.5  262.23  5007.8  261.45  5033.5  263.94
  5038.8  263.28  5064.5  265.78  5069.8  265.40  5095.5  268.14  5100.8  267.92
  5126.5  269.24  5131.8  268.90  5188.5  270.40  5241.4  270.96  5299.7  272.16
  5400.1  272.04  5479.9  271.25  5606.4  271.53  5649.5  272.40  5777.0  273.26
#Mann=5,-1,0
  4540.5    0.05       0  4813.2     0.1       0  4975.9    0.07       0
  4988.3     0.1       0  5241.4    0.05       0
Bank Sta=4975.9,4988.3
Exp/Cntr=0.3,0.1

Type RM Length L Ch R = 1,5885,192,192,192
BEGIN DESCRIPTION:
Mapping XS 841e363e
END DESCRIPTION:
XS GIS Cut Line= 2
      2120666.59     13400426.68      2119812.45     13400464.88
#Sta/Elev= 30
  4593.8  269.37  4664.2  269.27  4745.5  268.38  4812.1  267.37  4865.7  265.96
  4885.7  265.21  4891.3  264.80  4896.3  264.83  4925.7  263.79  4945.7  263.37
  4965.8  263.27  4975.8  261.63  4989.6  259.93  4990.1  259.13  5001.5  259.13
  5002.0  259.93  5005.8  260.96  5015.8  262.69  5035.8  264.92  5065.9  266.31
  5095.9  268.19  5113.3  269.01  5118.3  269.05  5145.9  270.69  5176.0  271.96
  5226.0  272.86  5256.1  273.89  5296.1  274.36  5406.2  274.37  5448.8  273.97
#Mann=4,-1,0
  4593.8    0.05       0  4812.1     0.1       0  4989.6    0.07       0
  5002.0     0.1       0
Bank Sta=4989.6,5002
Exp/Cntr=0.3,0.1

Type RM Length L Ch R = 1,5693,229,229,229
BEGIN DESCRIPTION:
Mapping XS a6bb7638
END DESCRIPTION:
XS GIS Cut Line= 2
      2120694.39     13400232.24      2119629.17     13400305.10
#Sta/Elev= 30
  4565.4  269.44  4594.9  269.29  4634.9  270.02  4735.2  269.02  4785.3  267.59
  4815.4  267.34  4847.4  266.22  4875.5  265.69  4945.7  263.13  4965.7  263.23
  4971.5  262.81  4999.6  259.31  5000.1  258.51  5011.5  258.51  5012.0  259.31
  5015.8  259.37  5035.9  262.51  5045.9  263.61  5055.9  264.31  5146.1  268.02
  5176.2  268.25  5226.3  269.08  5246.4  269.73  5263.3  269.89  5268.3  270.31
  5396.7  271.39  5446.8  272.43  5547.1  273.46  5567.1  273.85  5633.1  274.11
#Mann=4,-1,0
  4565.4    0.05       0  4847.4     0.1       0  4999.6    0.07       0
  5012.0     0.1       0
Bank Sta=4999.6,5012
Exp/Cntr=0.3,0.1

Type RM Length L Ch R = 1,5464,273,273,273
BEGIN DESCRIPTION:
UNT 006 in La Jarita Watershed 2.0
END DESCRIPTION:
XS GIS Cut Line= 3
      2120733.47     13399931.88      2120275.00     13400075.00
      2119598.66     13400231.06
#Sta/Elev= 30
  4515.4  268.38  4524.3  269.11  4534.7  269.07  4546.6  268.20  4566.2  267.60
  4606.3  267.58  4709.0  268.53  4786.2  268.12  4914.5  264.36  4941.7  263.11
  4946.9  263.26  4974.2  261.00  4979.4  261.42  4986.9  259.64  4987.4  258.84
  4998.8  258.84  4999.3  259.64  5014.5  261.63  5019.6  260.91  5026.5  261.98
  5047.0  263.17  5105.2  264.55  5201.0  266.23  5272.8  265.78  5308.7  266.58
  5328.7  266.64  5406.2  267.78  5590.9  272.41  5601.2  272.98  5689.8  273.80
#Mann=5,-1,0
  4515.4     0.1       0  4986.9    0.07       0  4999.3     0.1       0
  5308.7    0.05       0  5328.7     0.1       0
Bank Sta=4986.9,4999.3
Exp/Cntr=0.3,0.1

Type RM Length L Ch R = 1,5191,372,372,372
BEGIN DESCRIPTION:
Mapping XS 5ca1ac4e
END DESCRIPTION:
XS GIS Cut Line= 2
      2120395.95     13399786.91      2119541.73     13400196.65
#Sta/Elev= 30
  4865.2  268.54  4888.4  268.59  4910.6  267.91  4940.0  266.29  4955.0  265.18
  4962.7  264.57  4985.3  261.34  4990.9  259.54  4993.1  258.46  4993.6  257.66
  5005.0  257.66  5005.5  258.46  5008.0  258.62  5013.5  259.79  5036.2  262.68
  5058.8  263.32  5149.4  263.06  5172.1  263.67  5290.9  264.49  5308.0  264.39
  5336.2  264.79  5388.4  264.37  5417.8  264.65  5432.4  265.25  5465.2  265.77
  5576.1  269.40  5598.3  269.79  5658.9  272.09  5704.2  272.90  5812.6  273.62
#Mann=5,-1,0
  4865.2     0.1       0  4993.1    0.07       0  5005.5     0.1       0
  5388.4    0.05       0  5417.8     0.1       0
Bank Sta=4993.1,5005.5
Exp/Cntr=0.3,0.1
