HEC-RAS study DOAK Br.prj: DOAK Br Base Level Engineering

--- DOAK Br.g01 (geometry) --- (continued)

Type RM Length L Ch R = 1,28453,768,768,768
BEGIN DESCRIPTION:
Mapping XS 28cdd790
END DESCRIPTION:
XS GIS Cut Line= 3
      2065488.27     13477303.22      2065394.97     13477552.74
      2065353.78     13478040.51
#Sta/Elev= 30
  4731.8  459.09  4757.9  458.65  4765.7  457.60  4776.4  457.42  4838.1  454.68
  4873.7  451.87  4915.2  450.39  4953.9  446.33  4959.3  446.31  4978.9  445.22
  4984.2  445.29  4989.9  443.41  4992.3  439.55  4993.1  438.75  5000.3  438.75
  5001.1  439.55  5001.8  439.55  5010.5  443.89  5020.5  445.35  5049.3  444.57
  5061.5  444.27  5090.8  444.88  5110.9  446.13  5151.0  447.32  5211.2  447.89
  5261.4  448.87  5341.7  449.46  5415.4  449.56  5422.0  449.83  5487.7  449.86
#Mann=4,-1,0
  4731.8     0.1       0  4992.3    0.07       0  5001.1     0.1       0
  5049.3    0.05       0
Bank Sta=4992.3,5001.1
Exp/Cntr=0.3,0.1

Type RM Length L Ch R = 1,27685,402,402,402
BEGIN DESCRIPTION:
Mapping XS 7d7b0115
END DESCRIPTION:
XS GIS Cut Line= 4
      2064810.08     13477134.89      2064689.62     13477353.01
      2064709.16     13477594.98      2064930.25     13477747.80
#Sta/Elev= 30
  4659.0  453.97  4699.8  452.76  4721.6  452.74  4737.6  451.85  4743.4  452.10
  4759.4  450.73  4773.4  450.26  4781.2  450.65  4786.9  450.16  4808.7  449.98
  4840.8  447.98  4853.3  448.12  4876.2  447.48  4884.3  446.64  4897.8  446.37
  4930.2  445.37  4950.3  444.30  4980.4  444.31  4990.4  441.76  4996.1  438.07
  4996.9  437.27  5004.1  437.27  5004.9  438.07  5012.4  441.26  5020.5  444.57
  5060.7  442.84  5130.9  444.61  5176.8  445.06  5305.2  445.22  5419.7  446.08
#Mann=5,-1,0
  4659.0    0.05       0  4897.8     0.1       0  4996.1    0.07       0
  5004.9     0.1       0  5012.4    0.05       0
Bank Sta=4996.1,5004.9
Exp/Cntr=0.3,0.1

Type RM Length L Ch R = 1,27283,713,713,713
BEGIN DESCRIPTION:
Mapping XS 10099fa4
END DESCRIPTION:
XS GIS Cut Line= 4
      2064485.65     13477293.80      2064411.85     13477408.84
      2064429.21     13477818.99      2064480.64     13477906.85
#Sta/Elev= 30
  4609.2  445.55  4696.7  444.56  4727.1  445.15  4752.0  444.58  4802.1  443.76
  4822.1  443.12  4862.1  442.81  4882.2  443.01  4892.2  443.52  4922.2  443.82
  4937.9  443.51  4943.1  443.78  4952.2  443.57  4972.2  442.40  4982.2  441.10
  4992.3  439.12  4997.8  437.18  4998.7  436.38  5005.9  436.38  5006.7  437.18
  5012.3  440.12  5022.3  443.33  5032.3  443.78  5082.3  444.07  5122.4  445.25
  5216.4  445.86  5222.2  446.38  5232.1  446.49  5253.6  446.38  5258.2  445.89
#Mann=5,-1,0
  4609.2    0.05       0  4752.0     0.1       0  4943.1    0.05       0
  4997.8    0.03       0  5006.7    0.05       0
Bank Sta=4997.8,5006.7
Exp/Cntr=0.3,0.1

Type RM Length L Ch R = 1,26570,397,397,397
BEGIN DESCRIPTION:
Mapping XS 7a290a58
END DESCRIPTION:
XS GIS Cut Line= 4
      2064298.15     13477327.24      2063888.73     13477343.65
      2063868.45     13477504.32      2064298.11     13477772.53
#Sta/Elev= 30
  4518.8  443.89  4642.1  442.80  4757.6  442.85  4802.2  442.24  4832.2  442.70
  4837.3  442.13  4882.2  442.08  4892.3  441.49  4980.3  441.72  4990.4  440.91
  4992.4  434.40  4993.2  433.60  5000.5  433.60  5001.3  434.40  5010.5  438.77
  5020.6  440.97  5030.7  441.17  5050.9  440.16  5060.9  440.24  5082.1  441.47
  5088.3  442.38  5110.0  441.18  5160.5  442.55  5175.8  441.95  5197.0  442.59
  5254.8  441.99  5371.7  442.49  5458.9  442.62  5480.1  443.31  5597.0  444.81
#Mann=5,-1,0
  4518.8    0.05       0  4757.6     0.1       0  4992.4    0.07       0
  5001.3     0.1       0  5371.7    0.05       0
Bank Sta=4992.4,5001.3
Exp/Cntr=0.3,0.1

Type RM Length L Ch R = 1,26173,58,58,58
BEGIN DESCRIPTION:
Mapping XS 3cd9a47e
END DESCRIPTION:
XS GIS Cut Line= 6
      2064485.90     13477020.26      2063848.54     13477151.44
      2063674.93     13477209.60      2063546.46     13477252.13
      2063470.07     13477269.49      2063320.75     13477269.49
#Sta/Elev= 30
  4119.7  448.68  4262.8  444.39  4517.5  442.60  4710.7  441.39  4733.2  440.60
  4743.4  438.80  4769.7  438.34  4816.3  439.14  4825.2  440.43  4830.5  438.40
  4856.8  440.73  4862.1  438.30  4888.4  438.23  4893.6  437.10  4919.9  438.41
  4925.2  437.01  4942.9  438.06  4974.5  438.34  4983.2  436.49  4988.5  436.88
  4989.6  431.73  4990.1  430.93  5001.0  430.93  5001.6  431.73  5014.9  437.03
  5092.2  438.68  5110.8  439.75  5125.3  443.36  5151.9  445.39  5316.5  454.22
#Mann=4,-1,0
  4119.7    0.05       0  4517.5     0.1       0  4989.6    0.07       0
  5001.6     0.1       0
Bank Sta=4989.6,5001.6
Exp/Cntr=0.3,0.1

Type RM Length L Ch R = 1,26115,662,662,662
BEGIN DESCRIPTION:
Mapping XS 2fd3eb8a
END DESCRIPTION:
XS GIS Cut Line= 5
      2064439.03     13476991.62      2063850.28     13477072.44
      2063721.81     13477134.08      2063572.50     13477187.89
      2063312.99     13477213.07
#Sta/Elev= 30
  4166.5  447.57  4332.1  443.71  4502.5  442.49  4624.8  441.57  4655.1  440.01
  4669.7  441.49  4715.6  438.40  4725.7  440.35  4746.9  441.30  4766.6  439.11
  4780.8  439.65  4797.9  438.09  4811.0  440.71  4865.8  438.68  4871.4  440.22
  4888.5  438.76  4894.0  440.56  4898.7  438.99  4910.5  438.60  4931.8  439.96
  4985.0  437.08  4989.5  431.33  4990.1  430.53  5001.5  431.33  5005.0  436.83
  5010.3  437.77  5048.7  437.57  5099.6  440.39  5186.2  447.55  5322.7  453.97
#Mann=4,-1,0
  4166.5    0.05       0  4502.5     0.1       0  4989.5    0.07       0
  5001.5     0.1       0
Bank Sta=4989.5,5001.5
Exp/Cntr=0.3,0.1

Type RM Length L Ch R = 1,25453,348,348,348
BEGIN DESCRIPTION:
Mapping XS 5a45f9da
END DESCRIPTION:
XS GIS Cut Line= 4
      2064380.87     13476952.04      2063896.50     13476691.63
      2063486.78     13476686.42      2063343.41     13476860.88
#Sta/Elev= 30
  4249.8  446.73  4334.4  444.82  4523.8  442.87  4790.1  440.46  4797.7  439.67
  4831.2  439.93  4921.2  437.38  4932.0  436.10  4941.2  437.72  4971.3  437.42
  4981.3  433.04  4985.3  430.38  4985.8  429.58  4996.8  429.58  4997.3  430.38
  5001.3  433.05  5011.3  437.61  5021.3  439.10  5041.3  438.16  5071.3  438.22
  5108.9  440.51  5161.3  444.43  5191.3  445.77  5207.9  447.69  5217.1  447.38
  5252.3  448.85  5281.0  448.47  5330.5  449.56  5344.9  449.02  5435.3  450.57
#Mann=5,-1,0
  4249.8    0.05       0  4523.8     0.1       0  4985.3    0.07       0
  4997.3     0.1       0  5108.9     0.1       0
Bank Sta=4985.3,4997.3
Exp/Cntr=0.3,0.1

Type RM Length L Ch R = 1,25105,269,269,269
BEGIN DESCRIPTION:
Mapping XS bb66897c
END DESCRIPTION:
XS GIS Cut Line= 4
      2064111.77     13476665.57      2063844.42     13476406.91
      2063459.00     13476511.07      2063329.41     13476765.08
#Sta/Elev= 30
  4406.8  441.55  4716.1  438.73  4805.4  438.89  4850.7  438.03  4908.1  437.85
  4941.4  437.72  4946.5  436.99  4964.7  437.41  4975.0  436.55  4981.2  435.24
  4986.4  432.13  4989.7  429.11  4990.2  428.31  5001.2  428.31  5001.7  429.11
  5006.1  433.26  5015.9  437.03  5021.1  436.30  5037.2  438.13  5113.5  441.65
  5130.4  442.02  5170.3  444.57  5243.0  446.66  5281.9  448.82  5287.5  449.61
  5348.6  450.36  5376.4  451.39  5425.7  451.75  5459.7  451.70  5463.2  452.19
#Mann=7,-1,0
  4406.8     0.1       0  4805.4    0.12       0  4908.1    0.16       0
  4989.7    0.07       0  5001.7    0.16       0  5113.5     0.1       0
  5425.7    0.05       0
Bank Sta=4989.7,5001.7
Exp/Cntr=0.3,0.1

Type RM Length L Ch R = 1,24836,161,161,161
BEGIN DESCRIPTION:
Mapping XS d7955f11
END DESCRIPTION:
XS GIS Cut Line= 4
      2064181.25     13476655.20      2063875.67     13476226.35
      2063384.35     13476202.04      2063177.33     13476371.11
#Sta/Elev= 30
  4278.3  442.87  4300.5  442.22  4677.2  438.19  4865.6  439.16  4875.6  438.87
  4885.7  437.27  4937.1  435.99  4954.3  436.32  4965.8  436.85  4975.8  436.24
  4985.8  434.35  4989.8  429.28  4990.3  428.48  5001.3  428.48  5001.8  429.28
  5005.8  435.34  5015.8  437.35  5065.9  438.20  5095.9  436.94  5133.4  437.46
  5146.0  436.21  5166.0  437.62  5226.1  438.09  5249.1  439.31  5286.1  440.99
  5299.6  440.72  5312.4  442.01  5474.2  444.93  5483.2  445.69  5564.1  445.69
#Mann=7,-1,0
  4278.3    0.05       0  4300.5     0.1       0  4954.3    0.12       0
  4989.8    0.07       0  5001.8    0.12       0  5249.1    0.16       0
  5474.2    0.05       0
Bank Sta=4989.8,5001.8
Exp/Cntr=0.3,0.1

Type RM Length L Ch R = 1,24675,321,321,321
BEGIN DESCRIPTION:
Mapping XS 1e3566a8
END DESCRIPTION:
XS GIS Cut Line= 5
      2064541.34     13476740.04      2064228.82     13476330.30
      2063582.99     13476017.80      2063065.63     13476111.55
      2062809.34     13476302.03
#Sta/Elev= 30
  4002.7  452.22  4160.0  449.26  4445.1  440.83  4467.4  441.67  4481.9  440.27
  4568.4  438.87  4681.4  438.97  4794.3  437.20  4811.1  435.42  4822.5  437.35
  4907.3  438.60  4944.4  435.62  4975.0  436.07  4980.6  435.14  4991.6  429.71
  4992.1  428.91  5003.6  429.71  5011.1  434.18  5070.9  437.53  5093.5  435.78
  5263.9  438.56  5274.1  436.88  5294.4  439.23  5360.2  438.37  5579.0  444.97
  5642.7  448.25  5813.5  451.86  5919.2  452.59  6028.4  452.79  6080.6  454.23
#Mann=5,-1,0
  4002.7    0.05       0  4445.1     0.1       0  4991.6    0.07       0
  5003.6     0.1       0  5919.2    0.05       0
Bank Sta=4991.6,5003.6
Exp/Cntr=0.3,0.1

Type RM Length L Ch R = 1,24354,815,815,815
BEGIN DESCRIPTION:
Mapping XS f5f7b85f
END DESCRIPTION:
XS GIS Cut Line= 4
      2064901.10     13475888.89      2064151.13     13475875.00
      2063175.44     13475913.20      2062800.47     13475968.75
#Sta/Elev= 30
  3899.3  460.87  3985.4  458.00  4045.4  457.23  4085.4  455.49  4135.4  454.66
  4205.5  452.24  4565.5  443.92  4649.4  441.35  4685.6  439.35  4732.7  437.74
  4785.6  436.32  4955.8  435.90  4975.8  433.95  4985.8  434.34  4989.7  429.84
  4990.2  429.04  5001.4  429.04  5001.9  429.84  5005.8  430.82  5015.8  435.94
  5038.5  435.91  5105.9  436.23  5216.0  438.39  5291.4  437.66  5316.0  437.34
  5426.1  440.08  5747.6  450.08  5899.2  453.59  5939.7  453.97  6004.9  455.87
#Mann=6,-1,0
  3899.3     0.1       0  4732.7    0.12       0  4989.7    0.07       0
  5001.9    0.12       0  5038.5     0.1       0  5291.4    0.05       0
Bank Sta=4989.7,5001.9
Exp/Cntr=0.3,0.1

Type RM Length L Ch R = 1,23539,1230,1230,1230
BEGIN DESCRIPTION:
Mapping XS 9b801564
END DESCRIPTION:
XS GIS Cut Line= 3
      2064610.53     13475282.73      2063702.55     13475266.04
      2062771.21     13475386.22
#Sta/Elev= 30
  4090.1  452.77  4125.6  451.98  4155.6  452.22  4225.7  449.51  4365.7  446.14
  4375.7  445.11  4425.7  442.67  4435.7  443.24  4465.7  441.76  4485.7  441.64
  4625.7  437.55  4744.3  435.23  4805.8  434.22  4945.8  435.04  4965.8  434.18
  4975.8  432.97  4985.8  428.91  4988.4  426.39  4988.9  425.59  5000.1  425.59
  5000.6  426.39  5005.8  430.40  5015.9  433.49  5024.2  434.48  5086.5  433.40
  5154.2  434.04  5308.3  435.50  5422.1  437.49  5661.2  446.75  5937.3  454.46
#Mann=6,-1,0
  4090.1     0.1       0  4744.3    0.12       0  4988.4    0.07       0
  5000.6    0.12       0  5024.2     0.1       0  5154.2    0.05       0
Bank Sta=4988.4,5000.6
Exp/Cntr=0.3,0.1

Type RM Length L Ch R = 1,22309,1384,1384,1384
BEGIN DESCRIPTION:
Mapping XS 4a4b06ea
END DESCRIPTION:
XS GIS Cut Line= 4
      2064581.98     13474582.44      2064251.26     13474428.80
      2063269.49     13474392.34      2062503.11     13474530.25
#Sta/Elev= 30
  4046.9  441.04  4153.8  439.93  4193.8  438.57  4231.0  439.07  4417.8  435.24
  4577.9  433.26  4799.6  431.80  4968.2  432.76  4978.2  431.93  4992.1  425.77
  4992.6  424.97  5003.8  424.97  5004.3  425.77  5008.2  429.73  5018.2  431.30
  5048.3  432.54  5088.3  432.00  5108.3  430.21  5128.3  432.26  5168.2  431.26
  5348.2  434.04  5418.9  434.39  5662.5  439.81  5693.2  439.92  5713.5  441.76
  5764.4  441.70  5784.7  443.33  5805.0  442.56  5957.4  442.93  6172.7  447.19
#Mann=7,-1,0
  4046.9     0.1       0  4799.6    0.12       0  4992.1    0.07       0
  5004.3    0.12       0  5168.2    0.05       0  5348.2     0.1       0
  5662.5    0.05       0
Bank Sta=4992.1,5004.3
Exp/Cntr=0.3,0.1

Type RM Length L Ch R = 1,20925,1976,1976,1976
BEGIN DESCRIPTION:
Mapping XS 77159b3e
END DESCRIPTION:
XS GIS Cut Line= 4
      2064754.25     13473797.00      2064225.22     13473483.49
      2063230.43     13473197.03      2062749.54     13473328.12
#Sta/Elev= 30
  3974.6  442.74  4005.4  443.10  4048.2  441.49  4377.7  437.16  4463.4  433.67
  4498.3  434.06  4766.7  429.36  4915.4  431.03  4966.6  430.29  4974.8  428.09
  4979.1  422.53  4979.6  421.73  4991.4  422.53  4995.1  423.89  5000.3  422.88
  5006.0  428.37  5016.4  429.70  5118.2  430.34  5217.9  429.00  5266.2  425.92
  5285.3  428.60  5297.4  428.94  5318.2  427.97  5380.7  429.50  5487.9  429.68
  5734.1  432.27  5806.6  433.71  5824.2  435.03  5903.6  435.32  6123.2  439.86
#Mann=8,-1,0
  3974.6    0.05       0  4498.3     0.1       0  4915.4    0.12       0
  4979.1    0.07       0  4991.4    0.12       0  5118.2    0.05       0
  5487.9     0.1       0  5734.1    0.05       0
Bank Sta=4979.1,4991.4
Exp/Cntr=0.3,0.1

Type RM Length L Ch R = 1,18949,25,25,25
BEGIN DESCRIPTION:
Double Mapping XS 4591be85
END DESCRIPTION:
XS GIS Cut Line= 6
      2064823.73     13472616.47      2063833.21     13471930.56
      2063762.68     13471884.99      2063676.96     13471847.01
      2063466.45     13471841.58      2062949.98     13471950.00
#Sta/Elev= 30
  3591.0  438.59  3834.8  431.34  3864.5  431.53  3942.2  429.21  4209.8  426.23
  4410.4  425.98  4425.3  422.96  4446.2  422.23  4453.1  425.17  4467.2  425.43
  4547.6  425.52  4589.5  424.30  4598.3  425.23  4690.8  426.17  4828.6  426.74
  4868.7  425.68  4899.5  426.37  4915.0  425.16  4932.0  425.59  4937.5  424.46
  4962.3  423.83  4989.4  420.81  4989.9  420.01  5001.5  420.01  5002.0  420.81
  5065.7  422.93  5145.7  428.53  5384.4  432.08  5485.5  434.08  5712.0  437.13
#Mann=6,-1,0
  3591.0     0.1       0  4868.7    0.05       0  4989.4    0.04       0
  5002.0    0.05       0  5384.4    0.08       0  5485.5    0.05       0
Bank Sta=4989.4,5002
Exp/Cntr=0.3,0.1

Type RM Length L Ch R = 1,18924,759,759,759
BEGIN DESCRIPTION:
Double Mapping XS c12221b0
END DESCRIPTION:
XS GIS Cut Line= 6
      2064810.71     13472525.32      2063852.74     13471889.33
      2063687.81     13471829.65      2063632.47     13471816.63
      2063442.58     13471819.88      2062949.99     13471900.00
#Sta/Elev= 30
  3642.4  437.44  3782.9  434.03  3841.3  430.83  3985.3  428.50  4252.0  425.77
  4432.5  425.61  4441.5  425.21  4447.5  422.01  4453.5  421.91  4498.6  425.06
  4736.2  426.41  4814.6  425.29  4832.4  424.48  4896.2  426.39  4937.6  424.50
  4943.1  426.70  4972.2  425.91  4995.5  419.77  4996.0  418.97  5008.1  419.77
  5008.6  423.39  5013.8  426.51  5032.5  425.14  5079.1  427.25  5122.6  426.77
  5152.7  429.12  5289.9  430.68  5388.3  431.80  5488.4  433.66  5714.2  436.75
#Mann=7,-1,0
  3642.4     0.1       0  4814.6    0.05       0  4995.5    0.04       0
  5008.1    0.05       0  5289.9     0.1       0  5388.3    0.08       0
  5488.4    0.05       0
Bank Sta=4995.5,5008.1
Exp/Cntr=0.3,0.1

Type RM Length L Ch R = 1,18165,635,635,635
BEGIN DESCRIPTION:
Double Mapping XS 8ba2682b
END DESCRIPTION:
XS GIS Cut Line= 4
      2064893.17     13472486.27      2064169.58     13471570.32
      2063998.14     13471446.62      2062998.21     13471600.55
#Sta/Elev= 30
  3702.5  439.84  4022.7  428.58  4193.2  426.20  4584.3  424.40  4621.2  427.43
  4648.4  420.96  4670.9  418.98  4706.2  419.21  4720.6  421.55  4727.0  425.45
  4741.4  427.30  4766.9  425.05  4820.0  423.85  4867.4  425.23  4976.6  425.33
  4991.3  420.88  4992.4  417.13  4992.9  416.33  5005.0  417.13  5006.0  422.02
  5012.1  424.50  5030.9  424.63  5048.1  423.77  5071.0  424.91  5085.3  423.60
  5195.7  426.57  5438.5  429.38  5671.2  428.56  5752.7  430.10  6092.9  435.63
#Mann=7,-1,0
  3702.5     0.1       0  4766.9    0.05       0  4867.4    0.16       0
  4992.4    0.07       0  5005.0    0.16       0  5030.9     0.1       0
  5752.7    0.05       0
Bank Sta=4992.4,5005
Exp/Cntr=0.3,0.1

Type RM Length L Ch R = 1,17530,59,59,59
BEGIN DESCRIPTION:
Double Mapping XS 0334a8e9
END DESCRIPTION:
XS GIS Cut Line= 4
      2064975.61     13472473.23      2064647.01     13471401.05
      2064552.61     13471341.37      2062968.00     13471405.43
#Sta/Elev= 30
  3808.1  441.93  4256.0  427.21  4622.1  423.82  4663.9  418.33  4695.3  418.80
  4705.7  420.66  4712.8  424.55  4718.0  423.15  4726.7  427.38  4737.1  429.10
  4758.0  429.50  4778.3  423.87  4783.5  425.64  4789.4  422.93  4799.9  422.37
  4854.9  423.34  4984.9  424.12  4995.3  417.43  4995.8  416.63  5007.9  417.43
  5014.7  422.54  5048.8  425.64  5068.8  423.95  5339.0  424.73  5379.1  422.21
  5759.4  428.00  6009.6  429.71  6149.7  427.78  6259.8  429.59  6627.1  435.16
#Mann=6,-1,0
  3808.1     0.1       0  4854.9    0.05       0  4984.9     0.1       0
  4995.3    0.07       0  5007.9     0.1       0  6259.8    0.05       0
Bank Sta=4995.3,5007.9
Exp/Cntr=0.3,0.1

Type RM Length L Ch R = 1,17471,82,82,82
BEGIN DESCRIPTION:
Double Mapping XS a02d2ae7
END DESCRIPTION:
XS GIS Cut Line= 4
      2065023.35     13472438.49      2064676.31     13471352.22
      2064585.16     13471292.54      2062974.72     13471353.43
#Sta/Elev= 30
  3803.8  442.75  4195.9  428.04  4563.3  423.48  4633.9  426.93  4639.2  425.13
  4666.1  427.99  4689.3  428.46  4698.3  426.58  4703.5  428.61  4720.8  423.39
  4783.8  421.20  4831.5  423.29  4931.9  423.94  4980.2  423.68  4994.9  417.19
  4995.4  416.39  5007.5  417.19  5016.3  422.74  5022.3  423.87  5303.4  424.24
  5323.5  428.97  5383.5  420.64  5413.5  419.44  5443.5  420.84  5463.6  423.86
  5603.7  426.20  5973.9  429.00  6214.1  427.75  6310.8  429.48  6664.7  435.25
#Mann=6,-1,0
  3803.8     0.1       0  4831.5    0.05       0  4931.9     0.1       0
  4994.9    0.07       0  5007.5     0.1       0  6310.8    0.05       0
Bank Sta=4994.9,5007.5
Exp/Cntr=0.3,0.1

Type RM Length L Ch R = 1,17389,677,677,677
BEGIN DESCRIPTION:
Double Mapping XS 1f58a865
END DESCRIPTION:
XS GIS Cut Line= 4
      2065071.11     13472442.88      2064742.50     13471337.03
      2064656.78     13471238.29      2062953.05     13471301.34
#Sta/Elev= 30
  3788.7  445.46  3880.4  439.48  4068.2  433.33  4139.8  429.25  4276.8  428.57
  4569.5  423.26  4767.1  423.12  4788.0  421.32  4821.1  420.84  4845.6  423.98
  4921.0  422.95  4977.4  423.76  4984.8  422.02  4991.8  418.37  4992.3  417.57
  5004.7  418.37  5012.5  420.75  5041.0  423.12  5048.6  421.94  5072.0  423.33
  5335.1  423.63  5425.1  424.50  5485.2  426.88  5525.2  424.07  5715.3  427.26
  5915.5  426.78  6065.6  428.73  6409.4  428.50  6495.9  431.49  6778.0  435.17
#Mann=6,-1,0
  3788.7     0.1       0  4821.1    0.05       0  4921.0     0.1       0
  4991.8    0.07       0  5004.7     0.1       0  6409.4    0.05       0
Bank Sta=4991.8,5004.7
Exp/Cntr=0.3,0.1

Type RM Length L Ch R = 1,16712,1192,1192,1192
BEGIN DESCRIPTION:
Mapping XS 5412eec7
END DESCRIPTION:
XS GIS Cut Line= 4
      2065536.26     13471330.28      2065514.57     13471260.86
      2064455.54     13470815.98      2064312.36     13470805.14
#Sta/Elev= 30
  4120.8  425.77  4147.3  426.01  4203.9  424.68  4237.3  424.61  4432.6  422.85
  4480.1  421.82  4496.8  422.03  4527.6  420.84  4586.0  419.94  4648.6  421.76
  4681.0  420.07  4746.2  422.17  4768.6  421.61  4810.7  422.64  4969.5  422.59
  4984.9  421.03  4992.2  415.93  4992.7  415.13  5004.6  415.13  5005.1  415.93
  5006.5  418.01  5017.0  421.79  5022.4  422.42  5046.2  421.41  5190.9  421.67
  5234.3  420.93  5252.5  421.63  5276.2  421.35  5329.2  422.66  5485.8  424.77
#Mann=4,-1,0
  4120.8    0.05       0  4237.3     0.1       0  4992.2    0.07       0
  5005.1     0.1       0
Bank Sta=4992.2,5005.1
Exp/Cntr=0.3,0.1

Type RM Length L Ch R = 1,15520,82,82,82
BEGIN DESCRIPTION:
Mapping XS 810d4dfb
END DESCRIPTION:
XS GIS Cut Line= 4
      2065820.91     13470349.41      2065768.83     13470286.91
      2064734.98     13470148.89      2064399.99     13470350.00
#Sta/Elev= 30
  4295.4  422.74  4455.8  418.79  4532.0  418.32  4572.3  419.31  4642.9  416.71
  4663.1  418.39  4723.6  418.87  4730.0  420.65  4743.8  421.93  4753.9  420.80
  4764.0  417.86  4784.2  415.66  4848.3  412.53  4848.8  411.73  4860.7  411.73
  4861.2  412.53  4875.0  413.18  4895.1  415.77  4915.3  422.80  4925.4  423.13
  4945.6  421.16  4965.8  420.51  4975.9  415.55  4985.9  413.26  4996.0  413.49
  5016.2  420.28  5026.3  420.84  5359.2  418.43  5439.3  420.76  5810.5  423.68
#Mann=4,-1,0
  4295.4    0.05       0  4455.8     0.1       0  4848.3    0.07       0
  4861.2     0.1       0
Bank Sta=4848.3,4861.2
Exp/Cntr=0.3,0.1

Type RM Length L Ch R = 1,15438,290,290,290
BEGIN DESCRIPTION:
Mapping XS c1545bb4
END DESCRIPTION:
XS GIS Cut Line= 4
      2065919.87     13470320.76      2065794.87     13470200.97
      2064763.62     13470086.39      2064399.96     13470250.02
#Sta/Elev= 30
  4198.4  424.25  4454.5  419.11  4532.4  417.65  4650.0  419.86  4703.4  418.73
  4733.6  415.65  4740.6  417.25  4753.7  417.63  4773.9  421.39  4783.9  421.66
  4804.0  415.79  4824.7  413.89  4825.2  413.09  4837.6  413.89  4874.5  415.19
  4884.5  416.20  4894.6  419.14  4914.7  417.75  4944.9  422.42  4985.1  418.59
  4995.2  414.06  5012.3  420.62  5085.8  420.17  5102.8  418.50  5115.9  415.09
  5126.0  416.46  5136.1  419.85  5357.4  418.14  5473.4  420.79  5807.9  423.27
#Mann=4,-1,0
  4198.4    0.05       0  4454.5     0.1       0  4824.7    0.07       0
  4837.6     0.1       0
Bank Sta=4824.7,4837.6
Exp/Cntr=0.3,0.1

Type RM Length L Ch R = 1,15148,1028,1028,1028
BEGIN DESCRIPTION:
Mapping XS e24629b3
END DESCRIPTION:
XS GIS Cut Line= 4
      2065956.35     13470260.88      2065761.02     13470135.87
      2064695.91     13469966.60      2064529.63     13470018.56
#Sta/Elev= 30
  4092.6  424.20  4257.8  420.02  4307.9  420.14  4357.6  419.27  4452.1  417.23
  4583.7  419.39  4664.7  419.59  4674.9  418.18  4685.3  418.65  4705.2  415.57
  4725.5  416.43  4747.5  419.99  4766.0  419.50  4847.0  420.51  4897.6  419.77
  4928.0  420.54  4978.6  419.03  4990.0  413.23  4990.5  412.43  5002.4  412.43
  5002.9  413.23  5009.0  419.67  5120.4  418.79  5131.0  417.46  5140.6  418.46
  5160.9  418.85  5221.6  418.31  5241.9  417.51  5363.4  420.43  5577.2  421.62
#Mann=4,-1,0
  4092.6    0.05       0  4357.6     0.1       0  4990.0    0.07       0
  5002.9     0.1       0
Bank Sta=4990,5002.9
Exp/Cntr=0.3,0.1

Type RM Length L Ch R = 1,14120,837,837,837
BEGIN DESCRIPTION:
Mapping XS 17549d13
END DESCRIPTION:
XS GIS Cut Line= 3
      2066391.43     13469793.78      2065119.93     13469259.57
      2063950.03     13469303.72
#Sta/Elev= 30
  3456.6  425.64  3683.0  422.08  4086.6  417.26  4222.8  417.30  4233.7  416.74
  4245.4  412.66  4255.4  412.85  4263.7  416.37  4269.2  415.52  4287.5  417.23
  4483.2  415.77  4676.4  417.48  4734.7  416.35  4787.7  417.85  4960.8  416.71
  4980.8  415.25  4984.4  412.09  4984.9  411.29  4996.8  411.29  4997.3  412.09
  5010.8  415.18  5060.9  417.24  5160.9  415.24  5231.0  417.39  5455.7  418.81
  5631.3  420.11  5661.3  421.38  5671.3  420.44  5831.4  421.68  6006.5  421.30
#Mann=5,-1,0
  3456.6    0.05       0  3683.0     0.1       0  4984.4    0.07       0
  4997.3     0.1       0  5455.7    0.05       0
Bank Sta=4984.4,4997.3
Exp/Cntr=0.3,0.1

Type RM Length L Ch R = 1,13283,1474,1474,1474
BEGIN DESCRIPTION:
Mapping XS 4a640f26
END DESCRIPTION:
XS GIS Cut Line= 4
      2066394.10     13468652.35      2066182.31     13468562.08
      2064432.31     13468510.00      2064345.50     13468669.74
#Sta/Elev= 30
  3497.7  423.78  3547.2  422.44  3745.2  418.01  3865.3  417.55  4045.4  415.09
  4132.3  415.17  4145.4  414.08  4165.4  410.70  4175.4  415.32  4195.4  414.70
  4215.5  416.64  4225.5  416.63  4255.5  413.40  4295.5  414.42  4375.5  414.42
  4525.6  412.99  4625.6  414.81  4803.6  413.39  4845.7  414.30  4965.8  413.84
  4975.8  411.78  4979.3  409.96  4979.8  409.16  4991.7  409.16  4992.2  409.96
  4995.8  412.00  5005.8  413.90  5105.8  413.34  5369.3  415.03  5660.5  417.02
#Mann=5,-1,0
  3497.7    0.05       0  3547.2     0.1       0  4979.3    0.07       0
  4992.2     0.1       0  5369.3    0.05       0
Bank Sta=4979.3,4992.2
Exp/Cntr=0.3,0.1

Type RM Length L Ch R = 1,11809,119,119,119
BEGIN DESCRIPTION:
double Mapping XS 27c4fb58
END DESCRIPTION:
XS GIS Cut Line= 4
      2065619.48     13467448.96      2064464.19     13467350.70
      2064239.58     13467402.78      2064066.19     13467811.38
#Sta/Elev= 30
  3734.4  416.01  3939.6  412.12  4075.6  412.08  4100.2  408.10  4120.3  411.31
  4130.3  411.97  4290.9  411.23  4547.5  411.66  4612.0  411.19  4652.2  409.96
  4762.6  410.99  4913.6  410.92  4923.8  412.80  4932.0  416.24  4944.4  415.99
  4954.6  413.92  4974.7  406.55  5016.0  404.63  5016.5  403.83  5028.5  403.83
  5029.0  404.63  5065.1  407.24  5070.3  410.92  5077.8  412.86  5098.3  415.31
  5107.8  414.10  5118.9  410.01  5247.5  411.10  5333.4  412.56  5568.3  413.90
#Mann=4,-1,0
  3734.4     0.1       0  5016.0    0.07       0  5029.0     0.1       0
  5247.5    0.05       0
Bank Sta=5016,5029
Exp/Cntr=0.3,0.1

Type RM Length L Ch R = 1,11690,50,50,50
BEGIN DESCRIPTION:
double Mapping XS 646bf249
END DESCRIPTION:
XS GIS Cut Line= 5
      2065617.31     13467364.32      2064408.85     13467246.53
      2064320.96     13467276.91      2064239.58     13467294.28
      2064033.40     13467780.68
#Sta/Elev= 30
  3669.4  415.75  3953.1  411.48  4063.6  411.76  4103.8  408.90  4122.6  410.66
  4127.6  408.67  4133.9  410.31  4154.0  411.79  4214.3  410.67  4495.6  411.45
  4686.5  409.64  4867.4  410.62  4893.6  410.99  4908.8  414.42  4924.8  415.90
  4950.6  412.71  4961.7  407.76  4976.6  407.19  4989.6  408.79  4994.7  406.55
  5017.1  405.27  5017.6  404.47  5030.1  405.27  5054.3  406.43  5059.6  408.81
  5080.6  411.09  5093.2  414.76  5133.4  411.12  5250.0  411.36  5588.1  414.57
#Mann=4,-1,0
  3669.4     0.1       0  5017.1    0.07       0  5030.1     0.1       0
  5250.0    0.05       0
Bank Sta=5017.1,5030.1
Exp/Cntr=0.3,0.1

Type RM Length L Ch R = 1,11640,27,27,27
BEGIN DESCRIPTION:
double Mapping XS ba6be1b6
END DESCRIPTION:
XS GIS Cut Line= 5
      2065593.81     13467306.05      2064377.38     13467222.66
      2064234.15     13467246.53      2064192.92     13467319.23
      2064017.45     13467754.10
#Sta/Elev= 30
  3682.8  416.08  3932.2  411.45  4112.6  411.51  4122.6  410.94  4132.7  408.20
  4152.7  411.66  4232.9  410.29  4513.6  411.38  4673.9  409.63  4914.6  410.98
  4943.4  412.23  4948.4  414.38  4955.2  415.13  4975.5  413.68  4985.6  410.98
  4989.2  408.11  4989.7  407.31  5002.2  408.11  5004.2  410.67  5009.3  412.95
  5016.0  414.97  5026.2  415.43  5091.0  413.89  5096.8  412.10  5112.6  414.57
  5118.4  411.85  5158.7  410.24  5255.8  412.09  5320.4  411.47  5599.8  414.49
#Mann=4,-1,0
  3682.8     0.1       0  4989.2    0.07       0  5002.2     0.1       0
  5255.8    0.05       0
Bank Sta=4989.2,5002.2
Exp/Cntr=0.3,0.1

Type RM Length L Ch R = 1,11613,471,471,471
BEGIN DESCRIPTION:
double Mapping XS 5295d769
END DESCRIPTION:
XS GIS Cut Line= 4
      2065593.84     13467266.99      2064302.51     13467209.64
      2064189.66     13467231.34      2063969.65     13467728.51
#Sta/Elev= 30
  3675.1  415.94  3894.2  411.65  4094.4  411.51  4114.4  409.89  4124.4  410.02
  4134.4  411.77  4234.5  410.11  4281.5  411.12  4434.7  411.34  4594.8  410.83
  4674.9  409.46  4945.2  411.22  4985.5  410.51  4989.2  408.21  4989.7  407.41
  5001.7  407.41  5002.2  408.21  5016.1  409.31  5046.6  408.75  5056.8  410.08
  5067.0  410.28  5141.3  409.74  5151.3  410.30  5156.8  409.29  5174.1  409.51
  5185.6  410.95  5245.9  411.55  5302.0  412.46  5348.6  411.72  5626.3  414.72
#Mann=4,-1,0
  3675.1     0.1       0  4989.2    0.07       0  5002.2     0.1       0
  5245.9    0.05       0
Bank Sta=4989.2,5002.2
Exp/Cntr=0.3,0.1

Type RM Length L Ch R = 1,11142,30,30,30
BEGIN DESCRIPTION:
double Mapping XS 64ea674c
END DESCRIPTION:
XS GIS Cut Line= 5
      2065591.24     13467144.59      2064297.09     13466843.97
      2064231.98     13466817.93      2064082.24     13466787.55
      2063323.03     13467200.14
#Sta/Elev= 30
  3514.5  416.34  3578.2  414.24  3753.8  411.21  3900.8  410.85  3921.3  408.46
  3929.5  408.94  3934.6  411.54  4270.3  409.37  4504.2  409.94  4701.5  408.90
  4722.1  407.92  4775.4  409.14  4857.7  409.20  4881.9  407.74  4913.2  408.85
  4930.6  410.72  4940.8  410.43  4961.2  407.41  4985.3  406.64  4985.8  405.84
  4997.8  405.84  4998.3  406.64  5012.2  406.89  5032.6  410.75  5062.1  408.58
  5413.7  409.47  5511.7  410.85  5599.1  410.25  5746.4  412.16  5930.1  411.66
#Mann=4,-1,0
  3514.5     0.1       0  4985.3    0.07       0  4998.3     0.1       0
  5413.7    0.05       0
Bank Sta=4985.3,4998.3
Exp/Cntr=0.3,0.1

Type RM Length L Ch R = 1,11112,211,211,211
BEGIN DESCRIPTION:
double Mapping XS 259a2a8a
END DESCRIPTION:
XS GIS Cut Line= 4
      2065560.02     13467100.33      2064233.07     13466789.72
      2064059.46     13466750.66      2063270.62     13467064.90
#Sta/Elev= 30
  3559.1  415.83  3777.4  411.09  3867.5  411.19  3903.2  408.73  3915.1  411.06
  4005.9  411.06  4307.6  409.44  4591.3  409.66  4714.5  408.84  4735.1  407.55
  4790.3  409.18  4807.0  407.78  4875.3  408.70  4889.1  406.55  4930.2  410.93
  4985.2  406.42  4985.7  405.62  4998.2  406.42  5032.7  409.06  5057.8  409.55
  5073.7  408.55  5344.1  409.08  5363.0  409.33  5373.8  411.59  5384.5  409.42
  5412.4  409.35  5578.3  409.19  5675.2  411.05  5868.9  412.18  5949.0  411.29
#Mann=4,-1,0
  3559.1     0.1       0  4985.2    0.07       0  4998.2     0.1       0
  5412.4    0.05       0
Bank Sta=4985.2,4998.2
Exp/Cntr=0.3,0.1

Type RM Length L Ch R = 1,10901,18,18,18
BEGIN DESCRIPTION:
Double Mapping XS 897f5654
END DESCRIPTION:
XS GIS Cut Line= 4
      2065584.51     13466692.63      2064267.79     13466560.77
      2064077.90     13466569.45      2063265.40     13466991.99
#Sta/Elev= 30
  3597.2  421.48  3918.3  412.14  4018.8  410.89  4044.5  413.09  4069.1  407.99
  4089.2  410.80  4109.3  407.67  4139.4  407.78  4169.6  409.92  4179.6  413.43
  4199.7  409.74  4279.4  409.38  4320.3  409.34  4350.5  406.52  4360.5  409.15
  4712.3  408.35  4782.6  405.93  4812.8  407.84  4836.4  405.04  4836.9  404.24
  4849.4  405.04  4853.0  407.29  4883.1  406.45  4953.3  410.50  4973.4  406.53
  5013.4  405.89  5043.4  411.57  5083.5  406.94  5432.7  409.52  6026.4  411.53
#Mann=6,-1,0
  3597.2     0.1       0  4044.5    0.16       0  4279.4     0.1       0
  4836.4    0.07       0  4849.4     0.1       0  5432.7    0.05       0
Bank Sta=4836.4,4849.4
Exp/Cntr=0.3,0.1

Type RM Length L Ch R = 1,10883,32,32,32
BEGIN DESCRIPTION:
Double Mapping XS 3fb00cab
END DESCRIPTION:
XS GIS Cut Line= 4
      2065458.63     13466640.55      2064297.09     13466548.83
      2064125.65     13466545.58      2063192.55     13466955.51
#Sta/Elev= 30
  3725.5  417.91  3799.4  414.78  4033.7  410.37  4114.5  407.21  4170.5  409.60
  4180.5  413.52  4190.6  413.56  4200.6  410.17  4210.6  409.40  4266.9  409.41
  4321.0  406.67  4351.1  409.62  4401.2  408.36  4732.2  408.04  4782.4  406.05
  4812.5  407.76  4832.6  407.36  4836.1  404.51  4836.6  403.71  4849.1  404.51
  4852.6  407.02  4882.7  406.34  4982.8  411.29  4992.8  409.98  5032.8  411.09
  5076.2  407.01  5448.8  409.64  5587.1  408.85  5948.2  411.77  6081.3  410.86
#Mann=6,-1,0
  3725.5     0.1       0  4033.7    0.16       0  4266.9     0.1       0
  4836.1    0.07       0  4849.1     0.1       0  5448.8    0.05       0
Bank Sta=4836.1,4849.1
Exp/Cntr=0.3,0.1

Type RM Length L Ch R = 1,10851,1371,1371,1371
BEGIN DESCRIPTION:
Double Mapping XS 587843a5
END DESCRIPTION:
XS GIS Cut Line= 4
      2065423.89     13466575.44      2064272.13     13466516.28
      2064102.86     13466513.03      2063204.24     13466840.46
#Sta/Elev= 30
  3761.2  416.72  3880.2  415.38  4013.7  410.75  4063.9  409.92  4080.5  413.49
  4110.6  409.54  4243.5  408.90  4280.8  409.17  4300.8  406.16  4330.8  409.28
  4461.0  408.07  4691.3  408.53  4781.4  406.17  4801.5  407.70  4861.5  407.34
  4881.6  404.86  4891.6  407.51  4921.6  407.63  4971.6  406.81  4995.1  403.70
  4995.6  402.90  5008.1  403.70  5011.6  405.63  5021.6  406.95  5061.6  407.08
  5071.6  408.21  5156.0  407.19  5401.2  409.50  5496.6  408.60  6040.2  410.44
#Mann=6,-1,0
  3761.2     0.1       0  4013.7    0.16       0  4243.5     0.1       0
  4995.1    0.07       0  5008.1     0.1       0  5496.6    0.05       0
Bank Sta=4995.1,5008.1
Exp/Cntr=0.3,0.1

Type RM Length L Ch R = 1,9480,312,312,312
BEGIN DESCRIPTION:
Double  stream Mapping XS e00dd5e4
END DESCRIPTION:
XS GIS Cut Line= 4
      2065041.71     13465434.83      2064028.20     13465583.01
      2063623.20     13465766.74      2063046.69     13466570.08
#Sta/Elev= 30
  3833.0  418.49  3940.2  413.70  3981.3  413.52  4082.3  410.11  4112.6  410.45
  4173.3  408.17  4281.4  406.42  4567.4  404.89  4587.6  405.60  4678.6  404.42
  4696.0  404.97  4789.8  403.05  4959.6  405.16  4981.6  404.44  4996.6  402.66
  4997.0  401.44  4997.5  400.64  5009.5  400.64  5010.0  401.44  5019.7  403.62
  5058.5  404.43  5102.4  404.36  5124.3  405.32  5378.0  408.44  5656.8  409.58
  5833.5  408.88  6074.2  409.78  6116.0  408.95  6259.8  409.91  6290.8  410.00
#Mann=6,-1,0
  3833.0    0.05       0  3940.2     0.1       0  4997.0    0.07       0
  5010.0     0.1       0  5833.5    0.05       0  6259.8    0.08       0
Bank Sta=4997,5010
Exp/Cntr=0.3,0.1

Type RM Length L Ch R = 1,9168,309,309,309
BEGIN DESCRIPTION:
Mapping XS a635cc63
END DESCRIPTION:
XS GIS Cut Line= 4
      2064220.68     13465368.70      2063968.09     13465267.15
      2063672.52     13465448.14      2063010.31     13466450.17
#Sta/Elev= 30
  4534.0  408.11  4556.8  405.70  4581.0  404.70  4701.8  403.55  4821.6  403.59
  4902.6  404.54  4929.8  404.14  4966.5  406.07  4982.0  402.01  4987.8  401.60
  4990.3  399.29  4991.3  398.49  5003.5  398.49  5004.5  399.29  5009.2  401.14
  5018.7  401.28  5032.7  403.87  5040.0  404.29  5198.3  404.10  5388.0  407.29
  5589.6  408.62  5595.6  408.04  5619.5  408.13  5698.0  409.06  5740.1  408.49
  5776.2  409.14  5878.6  408.96  5884.6  409.60  6137.4  408.20  6353.9  409.17
#Mann=4,-1,0
  4534.0     0.1       0  4990.3    0.07       0  5004.5     0.1       0
  5619.5    0.05       0
Bank Sta=4990.3,5004.5
Exp/Cntr=0.3,0.1

Type RM Length L Ch R = 1,8859,69,69,69
BEGIN DESCRIPTION:
Mapping XS 9d55d323
END DESCRIPTION:
XS GIS Cut Line= 5
      2064995.62     13465286.35      2063871.53     13464969.52
      2063600.54     13465056.75      2063472.00     13465466.37
      2063010.19     13466309.73
#Sta/Elev= 30
  3398.9  417.16  3835.9  408.76  3863.3  412.81  3868.5  411.04  3897.3  417.54
  3902.5  415.86  3929.4  419.27  4048.9  415.71  4088.1  417.90  4156.2  416.36
  4161.4  418.39  4268.6  415.83  4307.8  418.14  4341.8  415.93  4381.0  418.28
  4454.3  416.15  4532.7  417.96  4565.9  416.95  4626.2  403.59  4666.8  402.94
  4834.4  403.90  4983.8  403.16  4999.7  399.15  5000.7  398.35  5013.9  399.15
  5048.6  402.72  5151.1  405.04  5287.8  405.20  5504.5  408.16  6242.3  408.10
#Mann=7,-1,0
  3398.9    0.05       0  4666.8     0.1       0  4834.4    0.05       0
  4999.7    0.04       0  5013.9    0.05       0  5287.8    0.08       0
  5504.5    0.05       0
Bank Sta=4999.7,5013.9
Exp/Cntr=0.3,0.1

Type RM Length L Ch R = 1,8790,887,887,887
BEGIN DESCRIPTION:
Mapping XS 304196e8
END DESCRIPTION:
XS GIS Cut Line= 5
      2065264.72     13464353.20      2064022.24     13464357.86
      2063545.20     13464966.69      2063432.35     13465409.40
      2062994.57     13466117.01
#Sta/Elev= 30
  2778.0  420.20  3407.7  413.53  3697.7  405.31  3785.2  405.00  3837.7  406.84
  3987.7  416.47  4016.6  412.53  4023.7  413.57  4030.0  411.47  4038.1  412.24
  4058.9  408.80  4067.0  409.38  4073.4  407.17  4087.8  408.09  4094.2  405.81
  4102.3  406.39  4108.7  404.14  4143.9  402.53  4423.2  401.49  4600.5  403.87
  4811.3  404.21  4957.3  402.70  5001.8  398.41  5002.8  397.61  5016.0  398.41
  5020.9  402.23  5061.8  404.20  5322.4  406.50  5370.9  406.98  6082.9  407.69
#Mann=7,-1,0
  2778.0    0.05       0  3785.2     0.1       0  4600.5    0.05       0
  5001.8    0.04       0  5016.0    0.05       0  5322.4    0.08       0
  5370.9    0.05       0
Bank Sta=5001.8,5016
Exp/Cntr=0.3,0.1

Type RM Length L Ch R = 1,7903,364,364,364
BEGIN DESCRIPTION:
Mapping XS 2c1b322b
END DESCRIPTION:
XS GIS Cut Line= 4
      2064968.54     13464262.82      2063413.84     13464274.70
      2063204.20     13464408.81      2062719.28     13465594.36
#Sta/Elev= 30
  3340.0  416.31  3573.6  413.40  3653.6  413.87  3972.2  405.77  4162.3  404.08
  4263.3  403.41  4507.9  401.37  4533.6  402.25  4606.2  400.93  4653.6  402.59
  4929.0  401.87  4975.8  399.22  4980.6  400.53  4988.3  396.55  4994.7  395.74
  4995.7  394.94  5008.9  395.74  5011.0  398.75  5024.0  402.16  5204.8  401.18
  5644.2  403.15  6023.2  403.33  6219.9  405.08  6260.9  407.09  6266.3  408.43
  6290.3  406.64  6367.8  406.48  6391.8  408.17  6397.2  406.49  6424.5  405.98
#Mann=12,-1,0
  3340.0    0.05       0  3972.2     0.1       0  4162.3    0.05       0
  4263.3     0.1       0  4507.9    0.05       0  4606.2     0.1       0
  4975.8    0.12       0  4994.7    0.07       0  5008.9    0.12       0
  5204.8     0.1       0  5644.2    0.05       0  6260.9     0.1       0
Bank Sta=4994.7,5008.9
Exp/Cntr=0.3,0.1

Type RM Length L Ch R = 1,7539,233,233,233
BEGIN DESCRIPTION:
Mapping XS e87ce57f
END DESCRIPTION:
XS GIS Cut Line= 4
      2064984.20     13463840.94      2063034.93     13464143.19
      2063040.14     13464453.09      2062588.93     13465511.42
#Sta/Elev= 30
  2915.7  415.40  3339.9  408.09  3451.2  409.08  3714.3  403.46  4004.4  403.11
  4005.6  403.12  4105.6  402.02  4220.3  401.64  4240.5  399.94  4278.0  401.57
  4301.3  397.90  4321.5  400.87  4362.0  401.79  4422.7  397.81  4442.9  401.75
  4503.6  400.55  4534.0  397.77  4554.2  400.97  4584.6  401.66  4968.1  400.39
  4980.1  400.25  4993.0  396.27  4994.0  395.47  5007.2  396.27  5020.7  400.41
  5110.1  398.79  5402.0  403.12  5883.4  402.87  6211.3  406.50  6348.7  405.65
#Mann=8,-1,0
  2915.7    0.05       0  4004.4     0.1       0  4005.6    0.05       0
  4105.6     0.1       0  4968.1    0.16       0  4993.0    0.07       0
  5007.2    0.16       0  5020.7     0.1       0
Bank Sta=4993,5007.2
Exp/Cntr=0.3,0.1

Type RM Length L Ch R = 1,7306,497,497,497
BEGIN DESCRIPTION:
Mapping XS 410ef7c0
END DESCRIPTION:
XS GIS Cut Line= 4
      2064895.59     13463710.74      2063006.29     13464066.37
      2062726.34     13464246.05      2062452.92     13465346.15
#Sta/Elev= 30
  2945.0  412.74  3108.4  411.75  3240.7  408.56  3375.8  409.34  3464.6  406.09
  3538.3  406.65  3643.2  403.66  3830.9  402.65  3891.9  400.31  3915.7  403.11
  3947.3  403.55  4003.4  402.53  4047.9  401.78  4390.5  401.77  4454.7  396.24
  4455.7  395.44  4468.9  396.24  4471.9  399.37  4492.3  401.82  4670.6  400.05
  4706.0  401.54  4910.9  400.70  4989.5  397.94  4997.9  399.20  5035.1  397.90
  5041.1  399.35  5047.2  398.05  5110.3  400.48  5302.1  402.59  6333.7  405.63
#Mann=8,-1,0
  2945.0    0.05       0  3947.3    0.08       0  4003.4    0.05       0
  4047.9     0.1       0  4454.7    0.07       0  4468.9     0.1       0
  4997.9    0.12       0  5110.3     0.1       0
Bank Sta=4454.7,4468.9
Exp/Cntr=0.3,0.1

Type RM Length L Ch R = 1,6809,67,67,67
BEGIN DESCRIPTION:
Mapping XS b587e5f6
END DESCRIPTION:
XS GIS Cut Line= 4
      2064859.14     13463611.77      2062672.95     13463692.67
      2062486.76     13463838.50      2062281.06     13464658.61
#Sta/Elev= 30
  2681.0  412.29  2805.2  411.74  2901.9  408.63  3005.4  409.00  3115.4  405.83
  3205.5  406.54  3515.7  402.02  3605.8  403.77  3664.4  401.99  3815.9  400.96
  3866.0  398.40  3876.0  400.52  4076.1  400.94  4136.1  399.94  4166.2  396.42
  4196.2  399.06  4286.2  400.49  4656.5  399.14  4676.5  400.60  4868.7  398.85
  4897.3  401.85  4904.2  401.42  4918.1  396.17  4933.5  394.41  4934.5  393.61
  4947.8  394.41  5122.2  394.94  5183.8  400.09  5505.9  403.02  5950.7  404.32
#Mann=5,-1,0
  2681.0    0.05       0  3664.4     0.1       0  4933.5    0.07       0
  4947.8     0.1       0  5183.8    0.05       0
Bank Sta=4933.5,4947.8
Exp/Cntr=0.3,0.1

Type RM Length L Ch R = 1,6742,109,109,109
BEGIN DESCRIPTION:
Mapping XS 9678e796
END DESCRIPTION:
XS GIS Cut Line= 4
      2064895.58     13463554.48      2062671.65     13463640.59
      2062463.32     13463757.77      2062213.34     13464559.69
#Sta/Elev= 30
  2612.9  413.30  2783.6  411.45  2873.7  408.49  2983.8  408.90  3083.8  405.70
  3173.9  406.78  3264.0  404.21  3504.1  402.23  3564.2  403.89  3618.9  402.30
  3814.4  400.47  3834.4  398.73  3894.4  400.98  4024.5  399.32  4084.6  400.32
  4094.6  398.33  4097.4  394.58  4098.4  393.78  4111.7  394.58  4114.6  397.52
  4144.6  400.61  4605.0  398.85  4645.0  400.74  4860.5  398.62  4919.8  402.05
  5106.0  403.12  5187.0  398.61  5211.7  399.30  5495.4  402.72  5917.5  403.65
#Mann=5,-1,0
  2612.9    0.05       0  3618.9     0.1       0  4097.4    0.07       0
  4111.7     0.1       0  5211.7    0.05       0
Bank Sta=4097.4,4111.7
Exp/Cntr=0.3,0.1

Type RM Length L Ch R = 1,6633,219,219,219
BEGIN DESCRIPTION:
Mapping XS 87154401
END DESCRIPTION:
XS GIS Cut Line= 5
      2064900.81     13463491.98      2062597.43     13463585.90
      2062497.17     13463613.24      2062256.29     13463778.61
      2062171.72     13464460.38
#Sta/Elev= 30
  2542.1  414.05  2828.1  408.17  2918.2  409.29  3028.3  405.42  3118.4  406.55
  3188.4  404.19  3537.8  402.71  3678.9  400.11  3778.9  400.66  3799.0  397.99
  3819.0  399.69  3879.0  397.32  3929.1  397.85  3949.1  400.51  4009.1  399.51
  4019.1  397.95  4022.0  395.00  4023.0  394.20  4036.3  395.00  4039.2  397.88
  4059.2  400.42  4870.6  399.20  4976.5  396.43  4997.5  396.44  5003.6  398.69
  5063.1  398.06  5075.3  400.59  5111.6  398.18  5241.8  398.73  5930.5  403.41
#Mann=5,-1,0
  2542.1    0.05       0  3537.8     0.1       0  4022.0    0.07       0
  4036.3     0.1       0  5241.8    0.05       0
Bank Sta=4022,4036.3
Exp/Cntr=0.3,0.1

Type RM Length L Ch R = 1,6414,470,470,470
BEGIN DESCRIPTION:
Mapping XS 6f589524
END DESCRIPTION:
XS GIS Cut Line= 4
      2064796.67     13463419.07      2062374.13     13463440.72
      2062002.97     13463752.51      2062109.18     13464408.69
#Sta/Elev= 30
  2487.4  411.70  2779.1  408.47  2879.1  405.40  2959.1  406.11  3199.1  403.04
  3289.1  404.29  3351.1  402.66  3549.1  399.74  3769.1  400.53  3789.1  398.82
  3799.1  400.27  3829.1  396.51  3869.1  398.44  3919.1  395.58  3929.1  396.35
  3939.1  399.74  3949.1  399.95  4149.1  398.26  4679.2  398.92  4859.2  397.90
  4907.1  395.94  4926.5  398.00  4975.9  397.60  4983.1  393.55  4984.1  392.75
  4997.4  393.55  5026.4  396.56  5068.3  397.90  5271.3  397.84  6059.5  402.58
#Mann=5,-1,0
  2487.4    0.05       0  3351.1     0.1       0  4983.1    0.07       0
  4997.4     0.1       0  5271.3    0.05       0
Bank Sta=4983.1,4997.4
Exp/Cntr=0.3,0.1

Type RM Length L Ch R = 1,5944,367,367,367
BEGIN DESCRIPTION:
Mapping XS 1749a99f
END DESCRIPTION:
XS GIS Cut Line= 4
      2064499.81     13463273.23      2062427.29     13463135.81
      2062081.16     13463033.81      2061469.31     13463163.70
#Sta/Elev= 30
  2755.5  408.10  2840.5  408.39  2960.8  404.70  3151.2  405.50  3275.4  402.82
  3612.2  399.04  3652.3  396.84  3752.5  399.13  3963.0  399.81  4003.0  395.19
  4015.8  399.40  4043.1  399.66  4073.2  394.75  4103.3  393.94  4143.3  398.79
  4166.5  399.16  4317.3  398.40  4353.8  395.43  4373.9  398.07  4980.9  396.84
  4990.4  395.76  4994.6  391.87  4995.6  391.07  5008.9  391.87  5043.5  396.68
  5142.8  397.06  5485.9  400.49  5639.3  399.18  5748.2  400.57  5818.9  400.70
#Mann=6,-1,0
  2755.5    0.05       0  3275.4     0.1       0  4994.6    0.07       0
  5008.9     0.1       0  5142.8    0.05       0  5748.2     0.1       0
Bank Sta=4994.6,5008.9
Exp/Cntr=0.3,0.1

Type RM Length L Ch R = 1,5577,323,323,323
BEGIN DESCRIPTION:
Mapping XS c4398a56
END DESCRIPTION:
XS GIS Cut Line= 4
      2064473.71     13463085.73      2062580.29     13462843.93
      2062292.75     13462747.36      2061449.97     13463050.01
#Sta/Elev= 30
  2894.2  411.12  3144.9  407.95  3253.0  404.16  3337.0  404.42  3749.8  400.33
  3850.6  396.67  3860.7  394.89  3931.3  398.02  4022.0  399.23  4415.2  398.58
  4425.2  397.37  4439.8  392.31  4465.6  398.51  4475.6  398.59  4519.6  396.25
  4526.1  397.81  4556.3  398.17  4616.8  394.98  4667.2  397.59  4909.2  395.86
  4935.2  393.50  4977.5  395.34  4987.9  393.03  4991.3  390.61  4992.3  389.81
  5005.6  390.61  5009.0  394.77  5019.6  396.92  5196.3  397.78  6001.8  399.71
#Mann=5,-1,0
  2894.2    0.05       0  3337.0     0.1       0  4991.3    0.07       0
  5005.6     0.1       0  5196.3    0.05       0
Bank Sta=4991.3,5005.6
Exp/Cntr=0.3,0.1

Type RM Length L Ch R = 1,5254,501,501,501
BEGIN DESCRIPTION:
Mapping XS 22599b6d
END DESCRIPTION:
XS GIS Cut Line= 4
      2064426.83     13462971.14      2062728.94     13462588.94
      2062368.70     13462557.47      2061350.01     13463049.99
#Sta/Elev= 30
  3079.6  412.15  3337.7  407.69  3360.7  405.24  3375.9  405.97  3475.9  405.90
  3557.8  404.62  4096.3  398.42  4157.8  395.46  4175.4  397.47  4229.5  398.64
  4373.0  397.08  4701.0  397.65  4844.0  396.07  4884.2  392.98  4914.3  396.07
  4954.4  396.27  4964.5  395.86  4987.4  390.96  4988.4  390.16  5001.8  390.96
  5064.9  396.04  5375.6  397.87  5420.8  397.04  5443.4  394.93  5460.5  397.50
  5466.0  396.58  5502.0  398.58  5827.5  397.92  6278.2  399.61  6313.1  400.01
#Mann=8,-1,0
  3079.6    0.05       0  3375.9    0.08       0  3475.9    0.05       0
  3557.8     0.1       0  4987.4    0.07       0  5001.8     0.1       0
  5502.0    0.05       0  6278.2    0.12       0
Bank Sta=4987.4,5001.8
Exp/Cntr=0.3,0.1

Type RM Length L Ch R = 1,4753,74,74,74
BEGIN DESCRIPTION:
Mapping XS d7cffdb8
END DESCRIPTION:
XS GIS Cut Line= 6
      2064184.49     13462693.28      2062642.57     13462222.83
      2062517.57     13462148.62      2062324.86     13462118.67
      2062195.96     13462119.97      2061188.62     13462933.63
#Sta/Elev= 30
  3162.1  408.22  3192.9  409.89  3336.6  406.45  3851.6  399.37  3977.1  398.96
  4027.1  397.10  4103.2  397.93  4154.8  396.23  4168.8  397.38  4217.5  396.39
  4239.6  394.54  4416.2  396.93  4740.3  395.91  4807.7  394.44  4879.8  393.91
  4942.4  387.91  5016.2  387.43  5017.2  386.63  5030.6  387.43  5084.1  387.60
  5134.4  391.36  5397.6  397.67  5432.8  396.48  5810.2  393.89  5866.2  395.62
  6066.2  396.70  6150.4  397.05  6239.7  397.47  6280.0  397.71  6538.4  399.78
#Mann=9,-1,0
  3162.1    0.05       0  3336.6     0.1       0  4807.7    0.12       0
  5016.2    0.07       0  5030.6    0.12       0  6066.2    0.05       0
  6150.4     0.1       0  6239.7    0.05       0  6280.0    0.12       0
Bank Sta=5016.2,5030.6
Exp/Cntr=0.3,0.1

Type RM Length L Ch R = 1,4679,92,92,92
BEGIN DESCRIPTION:
Mapping XS aab5bf28
END DESCRIPTION:
XS GIS Cut Line= 6
      2064192.51     13462523.23      2062663.41     13462179.87
      2062487.62     13462067.89      2062313.15     13462052.26
      2062145.18     13462101.74      2061202.93     13462825.31
#Sta/Elev= 30
  3166.5  412.49  3306.4  408.25  3983.9  398.71  4044.3  396.42  4147.9  396.70
  4189.7  394.36  4209.3  395.92  4233.0  394.88  4276.3  396.44  4701.3  395.74
  4750.8  400.17  4818.1  401.02  4966.1  401.41  5176.4  401.28  5209.2  400.69
  5220.1  398.74  5248.2  400.15  5253.5  398.31  5281.6  399.64  5286.8  397.64
  5330.4  396.32  5815.4  395.52  5872.5  393.70  5873.6  392.90  5886.9  393.70
  5935.9  396.53  6114.5  397.49  6188.8  398.34  6241.5  398.44  6480.4  399.58
#Mann=9,-1,0
  3166.5    0.05       0  3306.4     0.1       0  4818.1    0.12       0
  4966.1     0.1       0  5872.5    0.07       0  5886.9     0.1       0
  6114.5    0.07       0  6188.8     0.1       0  6241.5    0.12       0
Bank Sta=5872.5,5886.9
Exp/Cntr=0.3,0.1

Type RM Length L Ch R = 1,4587,499,499,499
BEGIN DESCRIPTION:
Mapping XS 0a3ca907
END DESCRIPTION:
XS GIS Cut Line= 6
      2064270.60     13462419.06      2062702.47     13462148.62
      2062552.73     13461998.88      2062327.47     13461953.30
      2062104.81     13462066.58      2061343.52     13462637.83
#Sta/Elev= 30
  3059.5  412.87  3116.9  413.50  3249.8  409.69  4019.1  396.45  4272.7  395.97
  4323.5  397.64  4348.6  396.20  4485.8  395.90  4536.6  396.35  4546.7  397.66
  4597.5  395.68  4864.7  394.20  4900.6  393.05  4957.9  394.60  4972.9  393.12
  4975.9  391.76  4976.9  390.96  4990.3  391.76  5003.5  393.38  5013.7  392.29
  5044.3  394.64  5207.8  394.72  5265.7  396.30  5742.2  394.82  5877.6  395.82
  5933.9  394.49  5983.8  396.28  6104.3  397.27  6251.6  398.92  6294.4  399.35
#Mann=8,-1,0
  3059.5    0.05       0  3249.8     0.1       0  4864.7    0.12       0
  4900.6     0.1       0  4975.9    0.07       0  4990.3     0.1       0
  6104.3    0.07       0  6251.6    0.12       0
Bank Sta=4975.9,4990.3
Exp/Cntr=0.3,0.1
