HEC-RAS study LAGUNILLAS Cr.prj: LAGUNILLAS Cr Base Level Engineering

--- LAGUNILLAS Cr.g01 (geometry) --- (continued)

Type RM Length L Ch R = 1 ,156540  ,605,605,605
BEGIN DESCRIPTION:
Mapping XS fb0fa72f
END DESCRIPTION:
XS GIS Cut Line= 5
      2042749.97     13518499.97       2042085.3     13517897.02
      2041998.49     13517831.92      2041891.07     13517717.99
       2041534.3     13517316.23
#Sta/Elev= 30
  3962.2  489.22  4345.5  485.96  4463.2  484.98  4474.7  484.86  4563.6  484.86
  4603.8  483.18  4670.4  480.71    4840  479.84  4889.6  477.94  4954.2   478.4
  4982.5  474.89  4986.4  469.31  4988.9  468.51  5006.9  469.31  5010.8  473.91
  5018.1  476.02  5046.3  478.12  5053.3   481.7  5060.2  479.61  5067.5  484.36
  5074.3   481.6  5081.6  485.57  5088.5  483.33  5095.8  485.95  5102.6  483.92
  5123.3  486.42  5130.8  485.36  5251.3  486.36    5365  484.77    5662   484.3
#Mann= 7 ,-1 , 0
  3962.2     .05       0  4345.5     .08       0  4463.2     .05       0
  4474.7     .08       0  4603.8     .05       0  4986.4     .04       0
  5006.9     .05       0
Bank Sta=4986.4,5006.9
XS Rating Curve= 0 ,0
Exp/Cntr=0.3,0.1

Type RM Length L Ch R = 1 ,155935  ,357,357,357
BEGIN DESCRIPTION:
Mapping XS 33fd90d1
END DESCRIPTION:
XS GIS Cut Line= 4
      2042872.83     13518508.91      2042517.16      13517891.6
      2042498.71     13517530.27      2041570.76     13517238.11
#Sta/Elev= 30
  4060.2  488.57  4244.9  486.44  4325.3  487.61  4341.1  486.33  4470.5  485.02
  4545.1  485.56  4588.3  484.39  4711.8   483.8  4772.6  484.47  4949.5  477.66
  4978.6  475.51  4989.3  467.93  4991.8  467.13  5007.3  467.13  5009.8  467.93
  5019.6  474.95  5039.6  477.21  5069.6  477.47  5119.7   475.6  5211.7  484.25
  5255.6  484.58  5285.1  485.26  5333.7  484.37  5366.1  485.02  5630.3  484.25
  5700.3  482.76  5737.9  483.97  5861.7     484  6029.3  485.87  6107.3  485.53
#Mann= 5 ,-1 , 0
  4060.2     .05       0  4978.6      .1       0  4989.3     .07       0
  5009.8      .1       0  5255.6     .05       0
Bank Sta=4989.3,5009.8
XS Rating Curve= 0 ,0
Exp/Cntr=0.3,0.1

Type RM Length L Ch R = 1 ,155578  ,395,395,395
BEGIN DESCRIPTION:
Mapping XS c013cfb0
END DESCRIPTION:
XS GIS Cut Line= 4
      2043102.01      13518357.9      2042896.93     13517682.18
      2042703.79     13517351.23      2041988.73     13516702.83
#Sta/Elev= 30
  4108.3  488.81  4268.1  485.97  4422.4  486.46  4455.3  485.25  4550.2  485.28
  4571.1  484.22  4686.1  483.39  4865.6  483.47  4938.6  481.45  4961.5  478.83
  4975.3  476.08    4983  475.41  4985.6  467.64  4988.4  466.84  5007.2  467.64
    5026  475.12  5047.5  476.63  5063.2  475.81  5112.2  477.42  5180.6  477.07
  5257.9  479.33  5332.1  483.15  5710.7  482.47  5760.7  481.47  5774.9  479.82
  5795.8  482.13    5831  483.93  6015.5  484.04  6114.1   487.6  6162.9  487.24
#Mann= 5 ,-1 , 0
  4108.3     .05       0  4975.3      .1       0  4985.6     .07       0
  5007.2      .1       0  5332.1     .05       0
Bank Sta=4985.6,5007.2
XS Rating Curve= 0 ,0
Exp/Cntr=0.3,0.1

Type RM Length L Ch R = 1 ,155183  ,475,475,475
BEGIN DESCRIPTION:
Mapping XS fe5af2a2
END DESCRIPTION:
XS GIS Cut Line= 4
      2043258.27     13518305.81      2043223.54     13517338.21
      2042832.91     13517107.09      2042273.89     13516436.03
#Sta/Elev= 30
  3822.7  488.77  4103.7   485.8  4273.8  486.24  4443.9  483.45    4594  483.63
  4694.1  479.72  4800.8  479.19  4886.8  475.15  4933.3  476.39  4982.4  475.02
    4998  468.26  4999.2  466.68  5001.9  465.88  5020.8  466.68  5025.2  475.11
  5040.9  474.56  5142.2  482.05  5200.8  484.43  5260.1   483.1  5535.5  483.12
  5656.5  481.11  5763.3  482.16  5820.2  484.46    5870  483.75    5926  487.02
  5968.9  486.83  6004.1  490.13  6047.1  489.81  6075.7  492.55  6118.2  492.88
#Mann= 5 ,-1 , 0
  3822.7     .05       0  4933.3      .1       0  4999.2     .07       0
  5020.8      .1       0  5260.1     .05       0
Bank Sta=4999.2,5020.8
XS Rating Curve= 0 ,0
Exp/Cntr=0.3,0.1

Type RM Length L Ch R = 1 ,154708  ,188,188,188
BEGIN DESCRIPTION:
Mapping XS 509e0947
END DESCRIPTION:
XS GIS Cut Line= 4
      2043445.77     13518071.44      2043442.72     13517410.91
      2043505.65     13517086.48      2042825.98     13516352.71
#Sta/Elev= 30
  4088.5  488.02  4384.9  484.67  4414.9  484.54  4464.9  486.01  4534.9  484.17
  4644.9  483.89  4734.9   479.2  4846.7  475.32  4970.6  474.53  4979.2  474.66
  4985.1  467.24  4987.8  466.44  5003.9  466.44  5006.7  467.24  5009.7  467.96
  5019.9  475.01  5030.1  476.34  5070.8  474.19  5109.1   474.3  5130.6  476.28
  5258.2  483.48  5328.5  483.23  5364.2  484.07    5398  482.25  5767.3  481.15
  5838.2  480.17  5915.9  481.43  6029.3   485.9  6050.2  485.25  6079.7  486.08
#Mann= 5 ,-1 , 0
  4088.5     .05       0  4970.6      .1       0  4985.1     .07       0
  5006.7      .1       0    5398     .05       0
Bank Sta=4985.1,5006.7
XS Rating Curve= 0 ,0
Exp/Cntr=0.3,0.1

Type RM Length L Ch R = 1 ,154520  ,1274,1274,1274
BEGIN DESCRIPTION:
Mapping XS a8eba8e9
END DESCRIPTION:
XS GIS Cut Line= 4
       2044211.4     13518279.79      2043804.37     13517310.72
      2043473.64     13516914.88      2042879.85     13516240.15
#Sta/Elev= 30
  3745.4  489.66  4236.5   488.7  4501.1   484.8  4760.4  483.39  4856.3  480.17
  4870.6   481.6  4921.2  478.83  4942.2  474.67  4977.4  474.74  4985.2  470.75
    4988  468.03  4988.5  467.55  4991.3  466.75  5007.5  466.75  5010.2  467.55
  5012.5  472.53  5020.3  475.86  5041.1  474.94  5063.2  475.84  5098.4   474.1
  5133.5  474.94  5155.6  474.01  5225.9  477.91  5268.9  479.12  5325.5   483.2
  5424.6   483.8  5456.6  482.13  5757.6  480.97  5863.8  479.62  6211.1   489.5
#Mann= 5 ,-1 , 0
  3745.4     .05       0    4988      .1       0  4988.5     .07       0
  5010.2      .1       0  5456.6     .05       0
Bank Sta=4988.5,5010.2
XS Rating Curve= 0 ,0
Exp/Cntr=0.3,0.1

Type RM Length L Ch R = 1 ,153246  ,488,488,488
BEGIN DESCRIPTION:
Mapping XS aea43c7a
END DESCRIPTION:
XS GIS Cut Line= 4
      2044841.61     13516878.76      2044616.77     13516434.57
      2044253.92     13516131.61      2043299.98     13515982.92
#Sta/Elev= 30
  4299.1  486.62  4538.7  484.62  4545.3  483.04  4589.8  481.55  4612.1  481.55
  4617.7  483.74  4634.4  482.49    4640  483.76  4656.7  483.78  4684.5  482.35
  4819.2  480.65  4890.4  477.86  4968.6  471.08  4975.4  468.75  4978.8  465.69
  4981.6  464.89  5000.6  465.69    5004  470.87  5010.6  472.41    5060  472.78
  5082.1  475.99  5124.9  477.13  5174.5  481.14  5203.2  481.07  5339.4  479.46
  5674.1  481.25  5845.4  478.53  5925.4  480.68  5987.1  478.42  6235.1  484.83
#Mann= 4 ,-1 , 0
  4299.1     .05       0  4978.8     .07       0  5000.6     .05       0
  5203.2     .05       0
Bank Sta=4978.8,5000.6
XS Rating Curve= 0 ,0
Exp/Cntr=0.3,0.1

Type RM Length L Ch R = 1 ,152758  ,590,590,590
BEGIN DESCRIPTION:
Mapping XS 9a6026f9
END DESCRIPTION:
XS GIS Cut Line= 4
      2045398.91     13516571.47      2044895.41     13515967.55
      2044516.07     13515859.04       2043269.3     13515894.35
#Sta/Elev= 30
  3980.1  487.21  4193.7  485.65    4264  486.47    4428  484.49    4484  485.23
  4512.6  483.62  4732.6  479.99  4808.4   475.6  4818.8  473.81  4827.1  474.33
  4832.3  477.06    4850  479.13  4881.2  479.02  4913.8  476.41    4954  471.15
  4977.8  472.83  4984.7  465.08  4987.5  464.28  5006.5  465.08  5011.6  472.81
  5026.8  471.77  5089.6  473.47  5140.9  477.64    5182   479.9  5402.1  478.12
  5722.2  481.91  5952.3  477.98  5982.3  479.37  6102.4  479.55  6408.2   485.8
#Mann= 5 ,-1 , 0
  3980.1     .05       0  4913.8      .1       0  4984.7     .07       0
  5006.5      .1       0  5140.9     .05       0
Bank Sta=4984.7,5006.5
XS Rating Curve= 0 ,0
Exp/Cntr=0.3,0.1

Type RM Length L Ch R = 1 ,152168  ,157,157,157
BEGIN DESCRIPTION:
Mapping XS a243036f
END DESCRIPTION:
XS GIS Cut Line= 4
      2045508.27     13515784.99      2044898.88     13515345.16
      2044523.88      13515371.2      2043238.76     13515696.11
#Sta/Elev= 30
  4049.9  485.84  4066.3  485.92  4109.6  482.94  4331.6  480.62  4559.8  479.11
  4725.4  479.61  4781.9  477.25  4825.4   476.9    4853  474.36  4870.9  472.38
  4875.9  473.11  4915.6   470.7  4955.7  472.25  4975.7  471.08  4984.9  463.99
  4987.7  463.19  5006.7  463.99  5013.3  470.32  5018.3  470.25  5055.9  476.48
    5066  479.08  5106.1  478.17    5300  478.44  5494.8  481.11  5623.1  480.59
  5764.1  478.03  5905.1  477.93  5987.1  480.18  6233.3  481.67  6502.9  487.59
#Mann= 5 ,-1 , 0
  4049.9     .05       0    4853      .1       0  4984.9     .07       0
  5006.7      .1       0    5066     .05       0
Bank Sta=4984.9,5006.7
XS Rating Curve= 0 ,0
Exp/Cntr=0.3,0.1

Type RM Length L Ch R = 1 ,152011  ,640,640,640
BEGIN DESCRIPTION:
Mapping XS d0573819
END DESCRIPTION:
XS GIS Cut Line= 4
      2045674.97     13515628.76      2045039.52     13515274.58
      2044608.95     13515196.72      2043211.41     13515613.11
#Sta/Elev= 30
  3979.1  486.89  4002.4  487.19  4047.8  484.01  4321.3  480.19  4751.8  479.05
  4841.5   476.8  4884.3  472.11  4924.6  469.95  4975.4  471.68  4984.8  463.38
  4987.6  462.58  5006.6  463.38  5012.1  468.85  5026.2  471.67  5036.4     472
    5077  478.73  5091.3  478.25  5578.6  481.08  5701.3  477.84  5795.2  478.16
  5815.9  475.31  5821.2     477  5847.4  474.09  5892.7  475.56  5925.9  480.39
  5931.1  478.93    5959  478.13  6140.5   479.8  6337.8  481.89  6602.4  487.36
#Mann= 5 ,-1 , 0
  3979.1     .05       0  4884.3      .1       0  4984.8     .07       0
  5006.6      .1       0  5091.3     .05       0
Bank Sta=4984.8,5006.6
XS Rating Curve= 0 ,0
Exp/Cntr=0.3,0.1

Type RM Length L Ch R = 1 ,151371  ,651,651,651
BEGIN DESCRIPTION:
Mapping XS 532d4712
END DESCRIPTION:
XS GIS Cut Line= 4
      2045924.95     13515368.34      2045325.97      13514849.5
      2044981.35     13514675.02      2043639.19     13514961.92
#Sta/Elev= 30
  3999.1  486.69  4178.7  482.93    4647  477.85  4871.1  479.58  4941.3   475.7
  4950.3  474.87    4967  468.36  4983.2   468.2  4983.9  460.66  4986.7  459.86
  5005.7  460.66  5011.5  468.79  5017.1  470.02  5078.3  469.16    5173  477.65
  5229.3  477.99  5437.8  479.57  5613.8  476.32    5624   477.4  5680.2  474.04
  5917.3  476.67  5930.8  478.92  5966.8  478.47  5971.9  482.01  6011.2  480.14
  6016.3  482.96  6060.7  480.67  6065.8  482.89  6110.2  478.67  6550.3  484.46
#Mann= 5 ,-1 , 0
  3999.1     .05       0  4941.3      .1       0  4983.9     .07       0
  5005.7      .1       0  5229.3     .05       0
Bank Sta=4983.9,5005.7
XS Rating Curve= 0 ,0
Exp/Cntr=0.3,0.1

Type RM Length L Ch R = 1 ,150720  ,323,323,323
BEGIN DESCRIPTION:
Mapping XS 555c92f3
END DESCRIPTION:
XS GIS Cut Line= 4
      2046169.72     13514925.61      2045341.59     13514165.47
      2045041.24     13514177.62      2043586.36     13514811.05
#Sta/Elev= 30
    3755  485.78  4537.1  475.34  4615.4  475.19  4735.6   477.6  4882.5  478.71
  4925.7  475.04  4955.8  468.85  4965.8  468.49  4975.8  466.25  4985.1  460.03
  4987.9  459.23    5007  460.03  5015.8  469.14  5045.8   467.4  5099.6  474.37
  5155.9  477.74  5358.3  475.79  5486.4  478.64  5562.1   477.4  5585.5  474.95
    5601  476.16  5713.6  475.56  6004.5  479.11  6080.9  479.05  6092.4  478.01
  6146.3   480.5  6209.5  481.34    6299  480.01  6429.9     481  6766.5   485.6
#Mann= 5 ,-1 , 0
    3755     .05       0  4882.5      .1       0  4985.1     .07       0
    5007      .1       0  5099.6     .05       0
Bank Sta=4985.1,5007
XS Rating Curve= 0 ,0
Exp/Cntr=0.3,0.1

Type RM Length L Ch R = 1 ,150397  ,654,654,654
BEGIN DESCRIPTION:
Mapping XS 956a3c8b
END DESCRIPTION:
XS GIS Cut Line= 4
      2046216.57     13514842.25      2045391.07     13513852.97
      2045072.49     13513879.01      2043378.99     13514649.15
#Sta/Elev= 30
  3533.6  486.05  4193.6  476.14    4420  473.97  4541.1  475.38  4703.8  479.87
  4841.5  479.39  4918.5  478.52  4938.5  476.99  4948.6  475.25  4968.6   468.4
  4978.7  467.98  4987.8  459.65  4990.6  458.85  5009.7  459.65  5018.8  467.26
  5048.9  467.19  5101.3  470.72  5204.9  476.03  5478.1  474.06  5558.3  474.95
  5581.4  473.62    5599  475.17    5622  473.91  5679.1  474.33  5892.2  479.32
  5966.9  478.93  6064.6  480.87  6346.9  480.01  6731.8  485.22  7002.1  486.99
#Mann= 5 ,-1 , 0
  3533.6     .05       0  4841.5      .1       0  4987.8     .07       0
  5009.7      .1       0  5101.3     .05       0
Bank Sta=4987.8,5009.7
XS Rating Curve= 0 ,0
Exp/Cntr=0.3,0.1

Type RM Length L Ch R = 1 ,149743  ,514,514,514
BEGIN DESCRIPTION:
Mapping XS 8a22c8e7
END DESCRIPTION:
XS GIS Cut Line= 4
      2045992.62     13514331.84      2045276.49     13513431.09
      2044945.76      13513292.2      2044338.15     13513383.69
#Sta/Elev= 30
  3618.4  479.62    3721  477.15    4091  473.05  4198.4  474.66  4368.1  480.33
  4569.8  476.65  4682.1  477.02  4774.1  470.51  4879.9  465.74  4951.2   468.4
    4975  467.87  4986.3  461.81  4993.2  458.59  4996.1  457.79  5015.1  458.59
  5020.2  471.71  5027.9  475.67  5067.7  475.17  5148.8  474.63    5159  476.34
  5169.1  475.85  5177.2  473.42  5182.2  474.05  5219.6  467.74  5246.1  467.23
  5280.3  468.96  5310.1  472.88  5411.8  477.15  5543.2  477.53  5742.3  480.78
#Mann= 6 ,-1 , 0
  3618.4     .05       0  4569.8      .1       0  4986.3     .07       0
  4993.2     .07       0  5015.1     .07       0  5067.7     .05       0
Bank Sta=4993.2,5015.1
XS Rating Curve= 0 ,0
Exp/Cntr=0.3,0.1

Type RM Length L Ch R = 1 ,149229  ,526,526,526
BEGIN DESCRIPTION:
Mapping XS b2e93f7c
END DESCRIPTION:
XS GIS Cut Line= 4
      2046102.03     13514316.26      2045593.44     13513446.13
      2045366.87     13513042.49      2044399.47     13513097.46
#Sta/Elev= 30
  3820.1  481.82  4023.3  477.47    4477  474.18  4498.5  470.97  4611.3  471.18
  4696.8  475.21  4921.7  475.91  4937.7  474.96  4958.9  467.12    4981  464.31
    4986  457.78  4988.9  456.98  5007.9  457.78  5012.7  464.71  5018.7   466.4
  5073.7  468.91    5074  468.93  5180.9   472.7  5230.6  475.59    5443  479.21
    5632  473.52  5653.3   473.1  5683.3  466.97  5723.4  466.43  5753.5  468.71
  5772.1   473.7  5836.7  474.41  5913.7  478.21    6114  476.93  6259.8  480.57
#Mann= 11 ,-1 , 0
  3820.1     .05       0  4611.3      .1       0  4696.8     .05       0
  4958.9      .1       0    4986     .07       0  5007.9      .1       0
  5073.7     .12       0    5074      .1       0  5180.9     .05       0
    5632      .1       0  5836.7     .05       0
Bank Sta=4986,5007.9
XS Rating Curve= 0 ,0
Exp/Cntr=0.3,0.1

Type RM Length L Ch R = 1 ,148703  ,392,392,392
BEGIN DESCRIPTION:
Mapping XS df19ae9c
END DESCRIPTION:
XS GIS Cut Line= 4
      2046232.23     13514139.16       2045909.3     13512952.79
      2045646.28     13512925.02      2044461.36     13512993.33
#Sta/Elev= 30
  3631.2  481.38  4008.6  476.66  4473.6  474.67  4692.6  475.17  4792.9  473.64
  4855.7   468.7    4895  467.56  4925.4   467.8  4975.7  464.41  4981.6  461.02
  4984.8  456.67  4987.7  455.87  5006.7  456.67  5015.9  466.07  5056.1  467.21
  5092.1  472.03  5216.7  476.48  5487.1  478.18    5673   473.3  5697.4  472.21
  5732.8  466.82  5787.6   465.8  5807.6  467.02  5817.6  468.89  5837.7  475.27
  5877.7   473.7  5903.6  474.38    6028  478.73  6218.3  476.94  6312.1  478.53
#Mann= 8 ,-1 , 0
  3631.2     .05       0  4792.9      .1       0    4895     .12       0
  4984.8     .07       0  5006.7     .12       0  5092.1     .05       0
    5673      .1       0  5903.6     .05       0
Bank Sta=4984.8,5006.7
XS Rating Curve= 0 ,0
Exp/Cntr=0.3,0.1

Type RM Length L Ch R = 1 ,148311  ,270,270,270
BEGIN DESCRIPTION:
Mapping XS c732034d
END DESCRIPTION:
XS GIS Cut Line= 4
      2046336.39     13514019.34      2046124.32     13512853.01
      2046044.46     13512698.15       2044478.5     13512826.54
#Sta/Elev= 30
  3694.3  481.46  3942.6  477.89  4725.3  474.97  4821.7  472.33  4967.5  466.02
  4980.4  464.59    4986  456.68  4988.9  455.88  5007.9  456.68  5012.5  461.16
  5019.1  464.75  5052.9     468  5123.7  468.09  5189.7  470.55  5320.4  474.97
  5655.5  476.26  5725.7  477.76  5810.9  477.24  5896.3  474.55  5930.8  469.83
  5937.4  470.79  5956.5  468.07  5996.6  465.92  6058.7  468.34  6086.9  473.08
    6127  474.84  6149.9  474.33  6247.4  477.85  6518.3  476.43  6625.2  478.52
#Mann= 7 ,-1 , 0
  3694.3     .05       0  4821.7      .1       0    4986     .07       0
  5007.9      .1       0  5189.7     .05       0  5930.8      .1       0
  6149.9     .05       0
Bank Sta=4986,5007.9
XS Rating Curve= 0 ,0
Exp/Cntr=0.3,0.1

Type RM Length L Ch R = 1 ,148041  ,822,822,822
BEGIN DESCRIPTION:
Mapping XS 91fc2287
END DESCRIPTION:
XS GIS Cut Line= 4
      2047086.39     13513186.04      2046432.56     13512672.75
      2046108.35     13512489.16      2044508.86     13512677.77
#Sta/Elev= 30
    3956  483.74  4171.9  482.07  4335.5  478.12    4698  474.23  4776.6  475.67
  4872.3  473.84  4883.8  475.35  4899.7  477.35  4922.3  477.19  4953.1  470.99
  4958.9  471.09  4980.5  462.69  4984.3  455.23    4988  454.43  5008.5  455.23
  5012.3  463.15  5033.9  466.36  5160.9  467.43  5455.2   474.9  5777.4  475.27
  5846.5  476.33  5898.3  479.05  5918.4  476.07  5968.7  474.39  6014.6  470.04
  6076.6   465.4    6176  465.23  6273.9  468.37  6364.5  476.33  6770.4  476.09
#Mann= 9 ,-1 , 0
    3956     .05       0  4883.8      .1       0  4984.3     .07       0
  5008.5      .1       0  5160.9     .05       0  6014.6      .1       0
  6076.6     .05       0    6176      .1       0  6273.9     .05       0
Bank Sta=4984.3,5008.5
XS Rating Curve= 0 ,0
Exp/Cntr=0.3,0.1

Type RM Length L Ch R = 1 ,147219  ,218,218,218
BEGIN DESCRIPTION:
Mapping XS bb8f6454
END DESCRIPTION:
XS GIS Cut Line= 4
      2047428.33     13513042.58      2045918.24     13511947.49
      2045775.01     13512188.38      2044455.57     13512521.66
#Sta/Elev= 30
  3079.9  480.14  4342.1   475.5  4619.6  475.71  4634.3  468.93  4655.2  472.81
  4663.7  469.16  4669.9  474.02  4684.6  466.94  4690.8  472.36  4699.3  467.75
  4720.1  473.71  4734.8  467.55  4755.7  473.06  4770.4  468.33  4776.6   472.6
  4785.1  469.73    4806  474.26    4942  472.56    4982  466.26  4985.5  453.96
  4989.2  453.16  5009.7  453.96  5012.2  461.92    5019  464.84  5113.1  465.54
  5369.9   474.3    5765  465.08  5895.9   480.4  6205.4  473.28  6586.4  476.59
#Mann= 5 ,-1 , 0
  3079.9     .05       0  4342.1      .1       0  4985.5     .07       0
  5009.7      .1       0  5113.1     .05       0
Bank Sta=4985.5,5009.7
XS Rating Curve= 0 ,0
Exp/Cntr=0.3,0.1

Type RM Length L Ch R = 1 ,147001  ,404,404,404
BEGIN DESCRIPTION:
Mapping XS 4ddc7561
END DESCRIPTION:
XS GIS Cut Line= 4
        2046550.       13511650.      2045831.87     13511661.83
      2045621.37     13512067.64      2044281.93     13512382.78
#Sta/Elev= 30
  4041.6  476.71  4146.6   473.9  4686.7  473.95  4826.6  472.29  4966.2  468.42
  4976.4  465.72  4982.1  466.51  4986.3  455.07  4990.1  454.27  5010.9  455.07
  5011.2  461.42  5020.7  463.86  5101.4  463.12  5152.7   467.6  5175.6  469.41
  5222.8   466.6    5228  467.91  5270.4  464.11  5275.5  464.92  5295.4  463.94
    5429  465.78  5521.5  471.21  5583.1  473.42  5841.8  474.73  5879.1  473.51
  5884.2  474.42  5921.4  472.57  5926.6  473.75  5952.9   472.8    6593  482.01
#Mann= 5 ,-1 , 0
  4041.6     .05       0  4826.6      .1       0  4986.3     .07       0
  5010.9      .1       0  5152.7     .05       0
Bank Sta=4986.3,5010.9
XS Rating Curve= 0 ,0
Exp/Cntr=0.3,0.1

Type RM Length L Ch R = 1 ,146597  ,434,434,434
BEGIN DESCRIPTION:
Mapping XS 05f02a13
END DESCRIPTION:
XS GIS Cut Line= 4
      2046682.25     13511332.94      2045768.94     13511531.62
      2045245.93     13511742.12      2045152.62     13511874.49
#Sta/Elev= 30
  3687.9   474.5  3819.2  473.43  3879.5  471.55  3981.9  471.32  4038.9  472.23
  4196.8  474.42  4309.4  473.79  4382.9  475.43  4470.9  473.22  4597.7  471.88
  4637.6  472.55  4820.8  465.75  4896.3  466.39    4918  465.36    4961  465.69
  4990.6  459.69  4991.7  453.77  4995.6  452.97  5016.6  453.77  5020.1  461.66
  5025.7  463.89  5044.3     469  5049.7  468.72    5058   471.6  5062.6  471.68
  5068.5  471.79  5079.6  474.98    5098   477.4  5225.9  478.93  5348.3  478.34
#Mann= 6 ,-1 , 0
  3687.9      .1       0  4038.9     .05       0  4597.7      .1       0
  4991.7     .07       0  5016.6      .1       0  5062.6     .05       0
Bank Sta=4991.7,5016.6
XS Rating Curve= 0 ,0
Exp/Cntr=0.3,0.1

Type RM Length L Ch R = 1 ,146163  ,228,228,228
BEGIN DESCRIPTION:
Mapping XS 78311302
END DESCRIPTION:
XS GIS Cut Line= 4
      2046644.11     13511275.68      2045801.49     13511312.44
      2045107.04     13511297.24      2044819.24     13511453.05
#Sta/Elev= 30
  3795.8  473.55  3824.9  473.99    3925  471.78  4035.1  471.17  4115.2  471.83
  4157.8  473.25  4345.4  473.11  4475.6  474.02  4621.9  472.02  4715.7  472.53
  4750.7  471.29  4765.7  469.37  4805.8  466.58  4845.8  465.27  4855.8   464.2
  4895.8  463.74  4965.8  464.62  4975.8  463.12  4983.3  453.57  4987.3  452.77
  5004.3  452.77  5008.2  453.57  5015.8  462.15  5025.8  463.75  5062.3  474.57
  5075.8  477.34  5125.8  478.22  5332.4   477.3  5495.4  478.68  5661.1  478.17
#Mann= 6 ,-1 , 0
  3795.8      .1       0  4157.8     .05       0  4621.9      .1       0
  4983.3     .07       0  5008.2      .1       0  5062.3     .05       0
Bank Sta=4983.3,5008.2
XS Rating Curve= 0 ,0
Exp/Cntr=0.3,0.1

Type RM Length L Ch R = 1 ,145935  ,294,294,294
BEGIN DESCRIPTION:
Mapping XS 064d2780
END DESCRIPTION:
XS GIS Cut Line= 4
      2046631.01     13511227.94      2045862.25     13511173.55
      2045282.82     13511069.38      2045020.26     13511177.88
#Sta/Elev= 30
  3858.6  473.74  3934.8  473.22  3970.5  471.75  4045.1  471.87    4097   470.5
  4175.4  472.63  4305.7  473.54  4385.9  472.89  4526.3  473.54  4656.1  471.92
  4697.6  471.51  4778.9  472.83  4789.1  472.01  4816.7  467.85  4821.7  468.13
    4850  463.74  4875.4  462.24  4941.5   463.6  4961.8  463.26  4971.9  461.56
  4980.4  454.13  4984.4  453.33  5001.4  453.33  5005.3  454.13  5012.6  466.13
  5032.9  470.69  5073.4  473.48  5114.2  476.17  5350.7  476.49  5502.1  478.37
#Mann= 6 ,-1 , 0
  3858.6      .1       0    4097     .05       0  4656.1      .1       0
  4980.4     .07       0  5005.3      .1       0  5073.4     .05       0
Bank Sta=4980.4,5005.3
XS Rating Curve= 0 ,0
Exp/Cntr=0.3,0.1

Type RM Length L Ch R = 1 ,145641  ,311,311,311
BEGIN DESCRIPTION:
Mapping XS a0725c11
END DESCRIPTION:
XS GIS Cut Line= 4
      2046615.66     13511128.09      2045844.89     13510965.21
      2045413.03     13510798.11       2045124.4     13510956.53
#Sta/Elev= 30
  4053.9  473.73  4096.8  473.93  4136.3  472.02  4183.4  471.77  4269.2  470.63
  4299.9     472  4335.3  471.14  4453.2  473.77  4555.4  472.56  4759.8  472.85
  4826.6  471.73  4895.2  471.33  4927.4  472.44  4948.8  472.26  4959.5  471.05
  4965.9  466.13    4981  459.28  4983.4  453.13  4987.4  452.33  5004.4  452.33
  5008.3  453.13  5013.1  460.33  5020.5  462.26  5034.6  463.69  5050.4  463.04
  5152.5  464.75  5227.2  468.49  5298.4  474.07  5455.3  474.52    5634  477.49
#Mann= 6 ,-1 , 0
  4053.9      .1       0  4183.4     .05       0  4826.6      .1       0
  4983.4     .07       0  5008.3      .1       0  5227.2     .05       0
Bank Sta=4983.4,5008.3
XS Rating Curve= 0 ,0
Exp/Cntr=0.3,0.1

Type RM Length L Ch R = 1 ,145330  ,386,386,386
BEGIN DESCRIPTION:
Mapping XS 102dc86f
END DESCRIPTION:
XS GIS Cut Line= 4
      2046652.12     13510815.59      2045933.87     13510594.12
      2045291.51      13510683.1      2045011.53     13510878.43
#Sta/Elev= 30
  3972.7  473.44    4097  472.95  4168.5  471.01  4265.6  470.23  4513.8  472.53
  4824.1  472.24  4874.6  473.26  4884.7  472.44  4911.4  467.43  4916.5  467.73
  4925.1  465.61  4965.5  463.37  4975.6   462.1  4983.2  459.46  4983.3  452.15
  4987.3  451.35  5004.3  451.35  5008.2  452.15  5015.9  462.25  5046.2  461.75
  5086.6   464.6  5116.9  464.82  5137.4  466.03  5147.2  467.06  5167.4  467.19
    5238  471.87  5328.9  473.15  5429.5  473.24  5522.8     476  5714.2  477.68
#Mann= 4 ,-1 , 0
  3972.7      .1       0  4983.3     .07       0  5008.2      .1       0
  5137.4     .05       0
Bank Sta=4983.3,5008.2
XS Rating Curve= 0 ,0
Exp/Cntr=0.3,0.1

Type RM Length L Ch R = 1 ,144944  ,476,476,476
BEGIN DESCRIPTION:
Mapping XS 685e29dd
END DESCRIPTION:
XS GIS Cut Line= 4
      2046664.04     13510752.22      2045827.53     13510249.07
      2045311.04     13510353.23      2045029.49     13510597.96
#Sta/Elev= 30
  3835.2  474.07  3977.6  473.09    4067   470.5  4189.4  469.79  4219.2  470.44
  4254.2  469.88  4422.5  472.97  4502.1  471.81  4698.3  472.67    4721  472.11
  4956.8  474.97  4964.8   474.5  4969.9  472.86  4977.2  466.13  4985.1  452.32
  4989.1  451.52  5006.1  451.52    5010  452.32  5015.6  458.86  5028.2  461.71
    5043  462.23  5071.5   462.8  5099.6   461.5    5168  463.94  5201.6  465.87
  5269.6  471.73    5386  470.83  5577.7  474.27  5655.5  476.82  5711.3   477.2
#Mann= 4 ,-1 , 0
  3835.2      .1       0  4985.1     .07       0    5010      .1       0
    5043     .05       0
Bank Sta=4985.1,5010
XS Rating Curve= 0 ,0
Exp/Cntr=0.3,0.1

Type RM Length L Ch R = 1 ,144468  ,570,570,570
BEGIN DESCRIPTION:
Mapping XS da503910
END DESCRIPTION:
XS GIS Cut Line= 4
      2046652.14     13510690.59      2045488.99     13509921.38
      2044924.75     13510121.03      2044846.92     13510330.74
#Sta/Elev= 30
  3392.9   473.7  3509.4  473.66  3605.3  470.57  3719.7  469.85  3978.5  472.82
  4065.8   471.6  4324.6  472.02    4469  473.64  4607.5  471.77  4658.6  472.56
  4757.9  470.29  4834.1  466.36  4950.7  462.71    4972  459.99    4978  452.46
    4982  451.66  5002.9  452.46  5003.8     458  5021.4  461.92  5077.9  461.67
  5099.2  467.91  5114.1  466.97  5139.7  471.63    5145  470.07  5162.9  472.73
  5215.9   475.7  5263.3  476.67  5279.6  478.29  5364.4  476.09  5609.6  476.57
#Mann= 4 ,-1 , 0
  3392.9      .1       0    4978     .07       0  5002.9      .1       0
  5215.9     .05       0
Bank Sta=4978,5002.9
XS Rating Curve= 0 ,0
Exp/Cntr=0.3,0.1

Type RM Length L Ch R = 1 ,143898  ,525,525,525
BEGIN DESCRIPTION:
Mapping XS 9c57bd16
END DESCRIPTION:
XS GIS Cut Line= 4
      2045867.65      13510092.3      2045534.56       13509687.
      2044925.19     13509454.36      2044248.93     13509722.07
#Sta/Elev= 30
  4032.5  472.24  4274.6  473.07  4352.6  471.64  4530.1  472.39  4574.7   470.2
  4744.5  464.96  4845.6  463.56  4908.9  460.61  4938.9  461.56  4963.4  461.11
    4969  457.76  4972.3  451.78  4976.3  450.98  4993.3  450.98  4997.2  451.78
  4999.1   451.8  5006.2  460.45  5016.9  466.59  5023.8  472.48  5029.2  469.78
  5038.3  472.58    5124  473.19  5206.8   475.3  5295.6  475.41    5309  476.24
  5349.4  473.91  5465.8  474.18  5532.2  475.98  5725.8  476.59  5936.7  480.24
#Mann= 3 ,-1 , 0
  4032.5      .1       0  4972.3     .03       0  4997.2     .05       0
Bank Sta=4972.3,4997.2
XS Rating Curve= 0 ,0
Exp/Cntr=0.3,0.1

Type RM Length L Ch R = 1 ,143373  ,920,920,920
BEGIN DESCRIPTION:
Mapping XS b6edb9ba
END DESCRIPTION:
XS GIS Cut Line= 4
      2045930.13     13510118.31      2045680.39     13509707.84
      2045430.39     13509098.46      2044529.55     13509092.29
#Sta/Elev= 30
  4072.8  471.83    4289  471.61  4436.1  472.94  4486.4  472.73    4552  470.77
    4606  470.81  4696.9  467.94  4736.7  465.03  4848.9  463.62  4867.4  460.76
  4891.4   459.9  4950.2   460.1  4979.6  461.52  4988.7  456.96  4991.1  452.72
  4995.1  451.92  5012.1  451.92    5016  452.72  5021.1  461.55  5027.5  463.16
  5032.9  465.86  5056.9  467.51  5140.2  468.83  5477.3  470.83  5637.3  474.97
  5767.3  474.34  5877.3  475.87  5887.3  474.85  5917.3  475.64  6112.8  476.88
#Mann= 4 ,-1 , 0
  4072.8      .1       0  4991.1     .07       0    5016      .1       0
  5140.2     .05       0
Bank Sta=4991.1,5016
XS Rating Curve= 0 ,0
Exp/Cntr=0.3,0.1

Type RM Length L Ch R = 1 ,142453  ,337,337,337
BEGIN DESCRIPTION:
Mapping XS b2937d87
END DESCRIPTION:
XS GIS Cut Line= 4
      2046190.56      13510232.9      2046289.18     13509336.39
      2046126.42      13509132.4      2044513.45     13508998.53
#Sta/Elev= 30
  3998.3  472.09  4456.7  470.17  4780.9  469.45  4946.9  468.46  4961.3  465.99
  4967.7   459.9  4975.7  457.45  4977.7  450.78  4981.6  449.98  5002.6  450.78
  5004.3  456.82  5017.3  460.97  5025.3  461.37  5046.2  459.67    5075  460.63
  5081.4  459.33  5110.2  458.96  5172.6   459.2  5212.8  461.06  5252.9  459.76
    5273  460.49  5323.2  466.25  5390.9  465.97  5744.6  468.03  5764.7  469.01
  6075.7     470  6274.9  475.35  6356.7     474  6467.1  474.12  6779.7  476.45
#Mann= 6 ,-1 , 0
  3998.3      .1       0  4456.7     .05       0  4780.9      .1       0
  4977.7     .07       0  5002.6      .1       0  5390.9     .05       0
Bank Sta=4977.7,5002.6
XS Rating Curve= 0 ,0
Exp/Cntr=0.3,0.1

Type RM Length L Ch R = 1 ,142116  ,529,529,529
BEGIN DESCRIPTION:
Mapping XS 1de90a01
END DESCRIPTION:
XS GIS Cut Line= 4
      2046642.96     13508991.34      2046488.84     13508976.15
        2045400.       13508950.       2044461.4     13508962.07
#Sta/Elev= 30
    4517  479.18  4536.3  478.25  4636.6  475.44  4865.8  466.41  4885.8   466.5
  4935.8  469.59  4965.8  468.75  4975.8  463.13  4985.8  455.37  4993.3  450.89
  4997.3  450.09  5018.3  450.89  5025.8  459.36  5055.8  457.92  5085.8  460.26
  5105.8  458.38  5135.8  458.62  5155.8   459.9  5175.8  464.28  5215.9  466.71
  5384.3  468.44    5926  470.05    6006  471.73    6046  474.39    6136  475.27
  6236.1  473.34  6416.1   475.2  6516.1  474.68  6576.1  476.27  6699.7  477.37
#Mann= 5 ,-1 , 0
    4517     .05       0  4536.3      .1       0  4993.3     .07       0
  5018.3      .1       0  5384.3     .05       0
Bank Sta=4993.3,5018.3
XS Rating Curve= 0 ,0
Exp/Cntr=0.3,0.1

Type RM Length L Ch R = 1 ,141587  ,451,451,451
BEGIN DESCRIPTION:
Mapping XS eeccb3f8
END DESCRIPTION:
XS GIS Cut Line= 4
      2046872.84      13508545.4      2046512.71     13508366.34
      2045436.32     13508691.86      2044478.49     13508888.86
#Sta/Elev= 30
  3915.9  484.48  4108.3  479.24    4389  469.22  4545.5  465.23  4733.6  469.28
  4884.3   469.2  4917.2  465.33  4942.5  464.34  4955.4  459.58  4973.9  458.38
  4982.3  451.57  4986.3  450.77  5007.3  451.57  5015.7  456.29  5021.3  457.82
  5054.2  458.12  5092.4  465.16  5120.1  457.46  5125.3  459.54    5141  458.28
  5191.2  459.83  5203.7  462.34  5235.1  461.26  5245.5  464.47  5267.5  467.41
    5430  469.89  5546.1  468.76  5778.3  474.54  6125.6  473.48  6420.5  475.69
#Mann= 5 ,-1 , 0
  3915.9     .05       0    4389      .1       0  4982.3     .07       0
  5007.3      .1       0    5430     .05       0
Bank Sta=4982.3,5007.3
XS Rating Curve= 0 ,0
Exp/Cntr=0.3,0.1

Type RM Length L Ch R = 1 ,141136  ,557,557,557
BEGIN DESCRIPTION:
Mapping XS 6892d7ef
END DESCRIPTION:
XS GIS Cut Line= 4
      2046815.59     13508212.09      2046547.43     13508129.79
      2045386.41     13508207.92      2044685.36     13508300.62
#Sta/Elev= 30
  3782.2  482.81    4068  473.16  4245.5  464.64  4295.7  463.19    4466  468.93
  4672.4  468.18  4796.8  466.87  4883.9  461.24  4917.1  459.55  4937.1  459.67
  4955.8  457.96  4977.2  458.21  4984.7  450.17  4988.7  449.37  5009.7  450.17
  5017.3  458.22  5057.4  465.92  5087.4  463.81  5105.4  465.17  5110.5  464.38
  5137.6  465.38  5157.6  468.95  5167.6  469.58  5237.9  470.26  5288.3   470.1
  5298.4  471.45  5389.2     471  5773.7  473.36  5779.4  473.32  5933.5  474.77
#Mann= 8 ,-1 , 0
  3782.2     .05       0  4672.4      .1       0  4883.9     .12       0
  4984.7     .07       0  5009.7     .12       0  5237.9     .05       0
  5773.7      .1       0  5779.4     .05       0
Bank Sta=4984.7,5009.7
XS Rating Curve= 0 ,0
Exp/Cntr=0.3,0.1

Type RM Length L Ch R = 1 ,140579  ,1479,1479,1479
BEGIN DESCRIPTION:
Mapping XS 0cb3de2e
END DESCRIPTION:
XS GIS Cut Line= 4
      2046862.45     13507998.54      2046523.56     13507695.77
      2045481.89     13507680.58      2044664.71     13508040.12
#Sta/Elev= 30
  3762.6  483.61  4025.6  474.68  4174.4  472.73  4209.5  470.63  4235.6  472.27
  4435.6  463.73  4485.6  458.69  4515.6   460.2  4555.6  465.82  4627.2     467
  4799.3  466.22  4865.7  465.48  4891.6  463.48  4935.7  456.88  4965.7  457.07
    4983  450.15  4987.1  449.35  5008.4  450.15  5015.7  457.44  5035.7  459.08
  5075.7  468.63  5115.7  468.64  5135.7  466.71  5155.7  468.78    5224  468.94
  5235.7   470.1  5341.2  469.55  5609.1  471.08  5784.5  473.25  6151.6  475.08
#Mann= 10 ,-1 , 0
  3762.6      .1       0  4627.2     .05       0  4799.3      .1       0
  4891.6     .12       0    4983     .07       0  5008.4     .12       0
    5224     .05       0  5341.2      .1       0  5609.1     .05       0
  5784.5      .1       0
Bank Sta=4983,5008.4
XS Rating Curve= 0 ,0
Exp/Cntr=0.3,0.1

Type RM Length L Ch R = 1 ,139100  ,356,356,356
BEGIN DESCRIPTION:
Mapping XS ebeaed2b
END DESCRIPTION:
XS GIS Cut Line= 4
      2047060.36     13507706.91      2046680.39      13506518.6
      2046366.16     13506435.27      2044618.84     13507898.57
#Sta/Elev= 30
  3628.7  477.58    3957  472.89  4125.9  471.52    4185  472.37  4260.6  470.61
  4479.7  470.12  4533.6  471.44  4575.6  470.15    4678  470.59  4796.1  469.35
  4875.5   466.9  4954.3  468.27  4964.6  466.75  4982.9   451.1  4987.1   450.3
  5008.4   451.1  5024.2  458.03  5078.4  456.38  5104.6  459.72  5141.2  462.47
    5671   467.6  6011.6  465.76  6160.2  466.94  6181.2  468.58  6330.7  469.02
    6423  471.37  6619.8  471.06  6832.2  471.86  7373.5  474.42  7480.5  475.14
#Mann= 8 ,-1 , 0
  3628.7     .05       0    3957      .1       0  4982.9     .07       0
  5008.4      .1       0  5141.2      .1       0  6619.8     .05       0
  6832.2      .1       0  7373.5     .05       0
Bank Sta=4982.9,5008.4
XS Rating Curve= 0 ,0
Exp/Cntr=0.3,0.1

Type RM Length L Ch R = 1 ,138744  ,449,449,449
BEGIN DESCRIPTION:
Mapping XS d491777e
END DESCRIPTION:
XS GIS Cut Line= 4
      2047133.23      13506045.4       2046762.1     13506003.67
      2046256.46     13506311.83      2044519.33     13507914.61
#Sta/Elev= 30
    4363  483.88  4366.4  483.73    4499  475.97  4743.8  466.76  4932.2  465.66
  4967.3  462.87    4982  456.64  4984.4  450.04  4988.8  449.24  5010.6  450.04
    5013  456.24  5025.8  459.89  5045.7   456.2  5061.5   454.9  5068.4  456.55
  5098.2  460.02  5185.8  463.02  5309.3  465.92    5728  466.83    5990  465.08
    6379  469.58  6506.6  473.43  6590.6  472.44  6819.6  471.36  7403.9  474.89
  7589.2  475.44  7603.3  475.81  7624.8  480.44  7681.5  479.43  7692.2  476.94
#Mann= 10 ,-1 , 0
    4363     .05       0  4366.4      .1       0  4984.4     .07       0
  5010.6      .1       0  5045.7     .12       0  5068.4     .07       0
  5185.8      .1       0  6590.6     .05       0  6819.6      .1       0
  7403.9     .05       0
Bank Sta=4984.4,5010.6
XS Rating Curve= 0 ,0
Exp/Cntr=0.3,0.1

Type RM Length L Ch R = 1 ,138295  ,414,414,414
BEGIN DESCRIPTION:
Mapping XS a9c83329
END DESCRIPTION:
XS GIS Cut Line= 5
      2047117.64     13505982.91      2046894.48     13505886.48
      2046015.57     13505906.01      2045461.39     13505946.45
      2044565.53     13506378.76
#Sta/Elev= 30
  4047.3  484.39  4154.6   478.8    4160  479.99  4178.1  477.54    4207  477.27
  4429.9     466  4628.5  464.39  4669.2  463.94    4760   463.3    4800  458.73
    4840  457.79    4890  458.19    4920  459.92  4960.1  458.43  4970.1  456.64
  4976.8  448.92  4981.3  448.12  5003.3  448.92  5010.1  458.66  5030.1  463.34
  5040.1  465.32  5090.1  467.86  5300.4  466.04  5486.2  466.81  5585.1  469.02
  5876.8  470.25  6095.6  473.04  6238.5  473.87  6402.3   472.7  6719.9  475.65
#Mann= 8 ,-1 , 0
  4047.3      .1       0  4628.5     .12       0  4669.2      .1       0
  4976.8     .07       0  5003.3      .1       0  5486.2     .08       0
  5585.1      .1       0  6095.6     .05       0
Bank Sta=4976.8,5003.3
XS Rating Curve= 0 ,0
Exp/Cntr=0.3,0.1

Type RM Length L Ch R = 1 ,137881  ,506,506,506
BEGIN DESCRIPTION:
Mapping XS ff765618
END DESCRIPTION:
XS GIS Cut Line= 4
      2047116.83     13505890.73      2046897.63      13505636.8
      2046014.38       13505448.      2044982.21     13505597.49
#Sta/Elev= 30
  4060.3  484.39  4062.1  484.28  4115.4  483.57  4164.8  480.32  4221.8  479.24
  4426.2  466.78  4500.7  463.78  4735.9  463.74  4811.8  464.29  4838.2  465.91
  4861.3  464.54  4916.1  457.85    4950  454.74  4971.1  456.14  4978.3  449.17
  4982.8  448.37  5004.8  449.17    5012  455.21  5054.1  466.74  5073.4  468.52
  5134.7  468.84  5291.3  465.62  5510.7  468.42  5540.8  469.75  5550.9   468.2
  5645.4  469.41  5985.4  473.64  6147.3  477.06  6278.5  480.29  6341.9  479.86
#Mann= 8 ,-1 , 0
  4060.3     .05       0  4062.1      .1       0  4916.1     .07       0
  4978.3     .07       0  5004.8     .07       0  5510.7     .05       0
  5645.4      .1       0  6147.3     .05       0
Bank Sta=4978.3,5004.8
XS Rating Curve= 0 ,0
Exp/Cntr=0.3,0.1

Type RM Length L Ch R = 1 ,137375  ,491,491,491
BEGIN DESCRIPTION:
Mapping XS 03bf6a58
END DESCRIPTION:
XS GIS Cut Line= 4
      2047244.82     13505840.75      2046895.46     13505306.94
      2046324.71     13504924.99      2045664.47     13504868.32
#Sta/Elev= 30
  4031.2   485.5  4253.8  480.91    4419  475.34  4554.6  467.13  4667.3   463.1
  4858.8   462.1  4915.9  460.14  4958.5  455.22  4972.9  455.37  4981.4  449.57
  4985.9  448.77  5007.9  449.57    5009  453.42    5024  457.47    5054   455.2
    5075  460.16  5111.1  463.28  5132.1  455.29  5162.1  454.64  5211.2  456.77
  5240.2  462.35  5255.2  461.77  5283.4  464.02  5435.9  464.83  5711.1  476.68
  5763.6  475.94  5787.2  478.29  5831.3  478.66  5897.6  480.93  6018.6  481.42
#Mann= 6 ,-1 , 0
  4031.2     .05       0  4253.8      .1       0  4981.4     .07       0
  5007.9      .1       0  5711.1     .05       0  5831.3      .1       0
Bank Sta=4981.4,5007.9
XS Rating Curve= 0 ,0
Exp/Cntr=0.3,0.1

Type RM Length L Ch R = 1 ,136884  ,339,339,339
BEGIN DESCRIPTION:
Mapping XS 01817dfc
END DESCRIPTION:
XS GIS Cut Line= 4
      2047669.71      13505363.1      2047308.97     13505011.91
      2046521.21     13504538.82      2045868.87      13504540.2
#Sta/Elev= 30
  4144.6  482.18  4217.4  482.01  4252.6  479.47  4273.9  480.94  4309.2  478.76
  4556.7  473.67  4634.5  470.63  4769.4  465.35  4919.4  462.64  4932.6  459.93
  4946.6  455.23    4968  454.32  4970.3  448.31  4974.8  447.51  4996.8  448.31
  5004.9   452.1  5014.3  452.53  5026.3  456.26  5041.8  458.95  5072.6  459.07
  5078.8  457.66  5107.2  458.83  5219.8  460.61  5264.8  460.86  5354.7  463.14
  5753.2  465.41  6016.4  477.64  6083.2  479.53  6144.2  482.77  6219.3  484.16
#Mann= 10 ,-1 , 0
  4144.6     .05       0  4634.5      .1       0  4769.4     .16       0
  4970.3     .07       0  4996.8     .16       0  5107.2     .12       0
  5219.8     .16       0  5264.8      .1       0  6016.4     .05       0
  6144.2      .1       0
Bank Sta=4970.3,4996.8
XS Rating Curve= 0 ,0
Exp/Cntr=0.3,0.1

Type RM Length L Ch R = 1 ,136545  ,72,72,72
BEGIN DESCRIPTION:
Mapping XS e3b8bb33
END DESCRIPTION:
XS GIS Cut Line= 4
      2047950.96     13504852.69      2047455.35     13504632.02
      2046977.92     13504523.52      2045784.28     13504243.32
#Sta/Elev= 30
  4132.5  484.05  4361.9  481.11  4628.5     471    4634  468.35  4651.7  469.34
  4657.2  466.54  4682.3   467.4  4687.5  465.14  4724.6  466.65  4730.5  463.94
  4754.6     465  4819.9  462.56    4901  460.26    4920  456.78  4962.5  456.01
  4972.8  454.49    4980  449.53  4984.5  448.73  5006.5  449.53  5020.1  453.28
  5120.2  457.74  5220.4  459.33  5266.5  460.09  5320.7  459.95    5421  462.18
  5528.6  463.58  5783.9  465.48  6032.7  472.76  6159.1   476.7  6390.7  478.92
#Mann= 16 ,-1 , 0
  4132.5     .05       0  4724.6      .1       0  4754.6     .05       0
  4819.9     .08       0    4920     .05       0    4980     .04       0
  5006.5     .05       0  5020.1      .1       0  5120.2     .07       0
  5220.4      .1       0  5266.5     .05       0  5320.7     .08       0
    5421     .05       0  5528.6      .1       0  6032.7     .05       0
  6159.1      .1       0
Bank Sta=4980,5006.5
XS Rating Curve= 0 ,0
Exp/Cntr=0.3,0.1

Type RM Length L Ch R = 1 ,136473  ,444,444,444
BEGIN DESCRIPTION:
Mapping XS 62d738ad
END DESCRIPTION:
XS GIS Cut Line= 4
      2048091.59     13504680.82      2047316.46     13504538.71
       2046776.1     13504382.46        2045550.     13503982.93
#Sta/Elev= 30
  4027.6   491.7  4120.3  489.17  4219.7  483.75  4517.9  474.77  4617.3  472.32
  4715.5  470.11    4752  465.52  4757.1  467.35  4805.2  461.91  4810.3  464.05
  4816.1  463.02  4845.1   460.1  4850.3  461.94  4915.8  457.23  4917.6  456.98
  4922.7  457.99  4981.9  450.58  4986.4  449.78  5008.4  450.58    5015  453.24
  5067.6  456.83  5313.7  461.12  5451.4  462.87    5800   465.3  5959.9   468.6
    6066  470.77  6147.1  476.08  6399.5  475.58  6640.5  478.87  6667.7  477.95
#Mann= 13 ,-1 , 0
  4027.6     .05       0  4120.3     .08       0  4219.7     .05       0
  4517.9     .08       0  4617.3     .05       0  4816.1     .08       0
  4915.8      .1       0  4917.6     .05       0  4981.9     .04       0
  5008.4     .05       0  5313.7      .1       0  5451.4     .05       0
  5959.9      .1       0
Bank Sta=4981.9,5008.4
XS Rating Curve= 0 ,0
Exp/Cntr=0.3,0.1

Type RM Length L Ch R = 1 ,136029  ,822,822,822
BEGIN DESCRIPTION:
Mapping XS cd87aa13
END DESCRIPTION:
XS GIS Cut Line= 4
      2048086.39     13504456.87      2047535.65     13504109.02
      2046669.73     13504024.58       2045633.3     13503894.37
#Sta/Elev= 30
  4014.2  488.38  4082.1  486.71  4465.3  470.36  4619.1  467.48  4706.4  467.49
    4841  461.64  4907.4  459.14  4937.5  455.59  4957.6  456.76  4968.6  455.34
  4977.7  452.34  4984.6  447.03  4989.1  446.23  5011.1  447.03  5017.9  455.64
    5028  457.22    5038  454.91    5070  457.91  5088.2  457.11  5167.2  460.35
  5228.9  460.09  5339.4  462.89  5411.4  462.48  5610.9  466.51    5752  464.59
  5895.7  466.13    6004   469.2  6034.2  468.27  6212.4  472.36  6580.2  476.68
#Mann= 7 ,-1 , 0
  4014.2     .05       0    4841      .1       0  4984.6     .07       0
  5011.1      .1       0    5070      .1       0  5167.2     .16       0
  5411.4      .1       0
Bank Sta=4984.6,5011.1
XS Rating Curve= 0 ,0
Exp/Cntr=0.3,0.1

Type RM Length L Ch R = 1 ,135207  ,480,480,480
BEGIN DESCRIPTION:
Mapping XS 8a0d949b
END DESCRIPTION:
XS GIS Cut Line= 4
      2048268.67     13503738.11      2047791.72     13503416.75
      2047264.38     13503312.58       2046218.3     13503654.23
#Sta/Elev= 30
  4036.6  478.07  4372.9  469.88  4501.9  467.53  4618.6  467.08  4659.3  464.77
  4740.9  462.95  4832.6  458.47  4914.2   456.8  4958.8  453.24  4975.3  451.74
  4982.5     446    4987   445.2    5009     446  5009.4  450.66  5016.1  452.91
  5036.5  455.61  5048.4  455.59  5097.6  458.43  5169.9   460.5  5253.8  462.15
  5269.7   463.4  5274.9  462.88  5295.9  465.01  5333.4  462.79  5397.2  461.16
  5516.8  460.85  5625.7   462.4  5737.7  466.37  5981.7  464.91  6249.7  468.15
#Mann= 6 ,-1 , 0
  4036.6     .05       0  4958.8     .07       0  4982.5     .07       0
    5009     .07       0  5048.4     .16       0  5169.9      .1       0
Bank Sta=4982.5,5009
XS Rating Curve= 0 ,0
Exp/Cntr=0.3,0.1

Type RM Length L Ch R = 1 ,134727  ,234,234,234
BEGIN DESCRIPTION:
Mapping XS f995d7a7
END DESCRIPTION:
XS GIS Cut Line= 4
      2048388.46     13503456.85      2047744.39     13502922.94
      2047445.02     13502918.83      2046294.74     13503462.07
#Sta/Elev= 30
  3969.8  474.69  4108.3  472.58  4250.2  473.17  4519.8  469.28  4620.1  468.84
  4768.6  464.07  4889.7  458.67  4895.8  458.85  4935.8  452.76  4965.8   452.3
  4975.8   450.5  4982.5  445.88    4987  445.08  5009.1  445.88  5015.7  453.22
  5075.8  456.46  5108.5  456.58  5148.2  457.14  5274.8  460.74  5314.8     460
  5344.3   460.8  5365.9   459.6  5485.3  459.53  5502.5   458.6  5604.6   459.6
  5650.2  462.03  5672.9  461.69  5868.9  467.71  6167.7  464.56  6377.9  468.36
#Mann= 7 ,-1 , 0
  3969.8     .05       0  4889.7      .1       0  4982.5     .07       0
  5009.1      .1       0  5108.5      .1       0  5148.2     .16       0
  5344.3      .1       0
Bank Sta=4982.5,5009.1
XS Rating Curve= 0 ,0
Exp/Cntr=0.3,0.1

Type RM Length L Ch R = 1 ,134493  ,1062,1062,1062
BEGIN DESCRIPTION:
Mapping XS 3729f88b
END DESCRIPTION:
XS GIS Cut Line= 4
      2048883.31     13502706.86      2047843.69     13502776.18
      2047408.67     13502659.08      2046607.24     13501696.46
#Sta/Elev= 30
  3737.6  472.62  4006.5  466.51  4136.8  461.86  4166.9  457.84    4217  462.36
    4227  464.71  4257.1  459.29  4317.2  458.29  4337.2  459.48  4389.2  467.74
  4689.8  466.44  4803.7  464.64  4894.5  460.59  4923.5  459.04  4962.4  453.48
  4974.9  450.26  4979.6  445.88  4984.2  445.08  5006.6  445.88  5016.4  453.06
  5026.7  454.58  5038.2  455.65  5063.4  453.75  5302.5  460.33  5378.1  461.25
  5526.8  459.59  5832.4  461.71    5960  460.89  6215.2  466.09  6482.6  467.68
#Mann= 8 ,-1 , 0
  3737.6     .05       0  4894.5      .1       0  4962.4     .16       0
  4979.6     .07       0  5006.6     .16       0  5063.4      .1       0
  5302.5     .05       0  5526.8      .1       0
Bank Sta=4979.6,5006.6
XS Rating Curve= 0 ,0
Exp/Cntr=0.3,0.1

Type RM Length L Ch R = 1 ,133431  ,563,563,563
BEGIN DESCRIPTION:
Mapping XS 3079a64f
END DESCRIPTION:
XS GIS Cut Line= 4
      2048883.23     13502321.43      2048199.98     13501920.77
      2047593.21     13501709.83      2046513.49     13501597.49
#Sta/Elev= 30
  3897.3  470.05  4172.3  466.51  4301.1   466.5  4492.7  462.92  4625.6  462.62
  4683.5  464.81  4705.2  463.43  4783.8  461.33  4895.7  455.45  4927.6  453.37
  4970.5  452.82  4980.5  450.22  4982.7  444.64  4987.4  443.84  5005.2  443.84
    5010  444.64  5012.2  449.72  5022.1  451.82  5027.4   452.5  5054.6  452.13
  5107.5  455.56    5340  463.07  5390.3  463.94  5460.7  463.74  5623.3  460.55
  5762.3  459.42  5862.8  460.53  6086.7  465.22  6134.3  466.75  6417.3  469.47
#Mann= 6 ,-1 , 0
  3897.3     .05       0  4895.7      .1       0  4982.7     .07       0
    5010      .1       0  5054.6     .05       0  6086.7      .1       0
Bank Sta=4982.7,5010
XS Rating Curve= 0 ,0
Exp/Cntr=0.3,0.1

Type RM Length L Ch R = 1 ,132868  ,726,726,726
BEGIN DESCRIPTION:
Mapping XS 4573d6a3
END DESCRIPTION:
XS GIS Cut Line= 4
      2048924.96     13501795.43      2048533.04     13501495.74
      2047883.74     13501256.16      2046748.95      13501191.3
#Sta/Elev= 30
  4045.9  473.63  4124.2  472.73  4417.1  465.35  4739.7  461.75  4812.4  458.55
  4832.8  458.62  4848.2  458.57  4873.3  455.89  4878.6  456.65  4898.4   455.4
  4910.2  456.09  4928.8  453.69  4934.1  454.59  4974.2  451.02  4981.8  444.26
  4986.6  443.46  5009.2  444.26  5014.8  449.79  5020.1  450.25  5027.5  452.53
  5054.9  449.93  5144.7  455.32  5270.2  457.26  5360.3  462.55  5515.1  460.95
  5650.8  458.27  5740.9  458.57  5921.2  461.31  6226.2  469.35    6368  472.85
#Mann= 6 ,-1 , 0
  4045.9     .05       0  4832.8      .1       0  4981.8     .07       0
  5009.2      .1       0  5054.9     .05       0  6226.2      .1       0
Bank Sta=4981.8,5009.2
XS Rating Curve= 0 ,0
Exp/Cntr=0.3,0.1

Type RM Length L Ch R = 1 ,132142  ,562,562,562
BEGIN DESCRIPTION:
Mapping XS 9fef0de6
END DESCRIPTION:
XS GIS Cut Line= 4
      2049284.28     13501118.31      2048336.86     13500627.68
       2047713.6     13500634.63      2046659.65     13500946.35
#Sta/Elev= 30
    3647  467.82  4361.1  460.69  4693.5  465.52  4712.2  462.87  4830.6  456.67
  4915.8  450.79  4975.8  452.27  4985.8  450.34  4992.1  443.52  4996.9  442.72
  5019.5  443.52  5025.8  449.05  5035.8  451.21  5082.4  454.08  5125.8  457.08
  5215.8  455.91  5245.8  452.84  5265.8  455.71  5325.8  457.33  5497.3  457.23
  5544.3  456.05  5563.8  452.93  5602.3   453.6  5607.5  456.15  5635.6  454.74
  5640.8  456.46    5659  454.41    5878  461.95    6157  466.28  6436.3  473.96
#Mann= 6 ,-1 , 0
    3647     .05       0  4830.6      .1       0  4992.1     .07       0
  5019.5      .1       0  5082.4     .05       0    6157      .1       0
Bank Sta=4992.1,5019.5
XS Rating Curve= 0 ,0
Exp/Cntr=0.3,0.1

Type RM Length L Ch R = 1 ,131580  ,377,377,377
BEGIN DESCRIPTION:
Mapping XS f991527b
END DESCRIPTION:
XS GIS Cut Line= 4
      2049378.04     13500623.52      2048353.79     13500191.92
      2048037.38     13500065.62      2047232.25     13500061.03
#Sta/Elev= 30
  3723.8  467.78  4039.1  461.72    4389  459.57  4580.8  461.95  4662.9  461.88
  4686.6  462.59  4725.4  466.66  4768.8  460.99  4867.8   454.5  4941.6  450.52
  4953.1  447.96  4971.9  449.19  4977.3  447.21  4981.7  442.03  4986.6  441.23
  5009.2  442.03    5017   448.4  5025.8  449.69  5031.2  447.75  5054.3  450.11
  5079.7  451.72  5085.1  450.96  5108.5   452.2  5146.2  451.76  5163.3  453.82
  5168.6  452.84  5188.3  455.33  5218.3  456.44  5468.3  458.93  5981.1  468.88
#Mann= 5 ,-1 , 0
  3723.8     .05       0  4867.8      .1       0  4981.7     .07       0
  5009.2      .1       0  5054.3     .05       0
Bank Sta=4981.7,5009.2
XS Rating Curve= 0 ,0
Exp/Cntr=0.3,0.1
