HEC-RAS study MACHO CREEK.prj: MACHO CREEK Base Level Engineering

--- MACHO CREEK.g01 (geometry) --- (continued)

Type RM Length L Ch R = 1 ,37841   ,248,248,248
BEGIN DESCRIPTION:
MACHO CREEK 62.0
END DESCRIPTION:
XS GIS Cut Line= 3
        2086025.     13456125.03        2085825.       13454125.
      2084325.01       13453825.
#Sta/Elev= 30
    2981  406.86  3081.5   406.1  3352.9  401.18    3383  399.72  3604.1  396.79
  4197.1   393.9  4370.4391.5104  4440.8  389.84  4558.9   392.3  4769.9  392.74
  4830.2  390.99  4842.8  389.79  4845.2  388.55  4846.1  387.75  4855.5  388.55
  4870.4  392.96  4880.5  393.19  4960.9  392.96  4988.5  389.78  5021.6  389.53
  5052.2  391.82  5062.4  391.92  5072.6  390.27 5091.69391.5101  5113.4  393.35
  5164.4  392.16  5460.1  394.54  6000.6  395.26  6245.4  400.47  6520.7  409.39
#Mann= 3 ,-1 , 0
    2981      .1       0  4845.2     .07       0  4855.5      .1       0
Bank Sta=4370.4,5091.69
XS Rating Curve= 0 ,0
Exp/Cntr=0.3,0.1

Type RM Length L Ch R = 1 ,37593   ,430,430,430
BEGIN DESCRIPTION:
MACHO CREEK 61.0
END DESCRIPTION:
XS GIS Cut Line= 6
      2086467.94     13454719.09      2085955.76     13453986.42
       2085810.2     13453961.72      2085770.27     13453979.86
      2085510.39     13453967.58      2084653.81     13453743.97
#Sta/Elev= 30
  3931.8  393.58  4173.6  392.08  4295.7  389.44  4339.4  390.67  4352.4  389.75
    4376  391.02  4382.1  390.43 4384.02389.3347  4388.2  386.95  4397.8  385.45
  4398.7  384.65  4407.2  384.65  4408.1  385.45  4417.8  388.16  4424.8  391.46
  4533.8  390.86  4718.7  392.45  4868.1  391.78  4917.8  393.08  4958.4  392.45
  4973.4  391.35    4989  388.77  4994.5  388.49 4996.88389.3374  5011.9  392.76
  5132.6  391.05  5272.6  393.83  5882.4  394.41  6056.3  396.79  6162.7   399.4
#Mann= 3 ,-1 , 0
  3931.8      .1       0  4397.8     .07       0  4408.1      .1       0
Bank Sta=4384.02,4996.88
XS Rating Curve= 0 ,0
Exp/Cntr=0.3,0.1

Type RM Length L Ch R = 1 ,37163   ,244,244,244
BEGIN DESCRIPTION:
MACHO CREEK 60.0
END DESCRIPTION:
XS GIS Cut Line= 5
      2086543.76     13456485.27      2086561.12     13454419.32
      2086170.49     13453898.49      2085823.27     13453690.15
      2085540.89     13453560.78
#Sta/Elev= 30
  1767.8  403.49  2638.1  399.36  2708.1  397.81  2748.1  398.72  2988.1  397.79
  3138.1  396.01  3418.1  394.99  3448.1  393.76  3458.1  394.62  3558.1  394.29
 4073.92389.5774  4090.6  388.56  4126.7  383.79  4153.8  384.03  4179.8  383.99
  4319.4   384.3  4364.6  383.53  4365.5  382.73  4374.9  383.53  4434.3  383.56
  4448.9  385.41  4463.5  390.11  4469.7  390.65  4615.9  391.05  4775.2  389.69
  4937.8  390.49  4966.3  389.04 5001.54389.5777  5074.9   392.2  5200.4  392.37
#Mann= 6 ,-1 , 0
  1767.8      .1       0  4153.8     .05       0  4179.8      .1       0
  4319.4     .05       0  4364.6     .07       0  4374.9      .1       0
Bank Sta=4073.92,5001.54
XS Rating Curve= 0 ,0
Exp/Cntr=0.3,0.1

Type RM Length L Ch R = 1 ,36919   ,163,163,163
BEGIN DESCRIPTION:
MACHO CREEK 59.0
END DESCRIPTION:
XS GIS Cut Line= 4
      2086995.15     13455695.37      2086647.92     13454323.84
      2086170.49      13453759.6      2085775.48     13453449.85
#Sta/Elev= 30
  2565.5  398.63  3926.7  391.95  4024.1  394.08  4038.4  392.81  4044.9  394.11
    4067  392.94  4102.1  394.13  4116.4  392.72  4122.9   394.2  4130.7  393.06
  4137.2  394.21  4288.9  394.02  4290.6  394.06  4358.1  393.09  4421.8  395.38
    4535  393.85  4577.8  395.14  4641.5  394.23  4726.4  389.49 4811.59389.1362
  4818.9  387.97  4847.8  388.98  4863.4  387.01  4864.3  386.21  4873.7  387.01
    4883  388.51  4947.2  389.75  4982.5  387.68 5029.17389.1369  5221.4  391.89
#Mann= 5 ,-1 , 0
  2565.5      .1       0  4288.9     .05       0  4290.6      .1       0
  4863.4     .07       0  4873.7      .1       0
Bank Sta=4811.59,5029.17
XS Rating Curve= 0 ,0
Exp/Cntr=0.3,0.1

Type RM Length L Ch R = 1 ,36756   ,1652,1652,1652
BEGIN DESCRIPTION:
MACHO CREEK 58.0
END DESCRIPTION:
XS GIS Cut Line= 3
      2087081.94     13455669.29      2086760.77     13454306.47
      2085886.13     13453355.47
#Sta/Elev= 30
  2632.6   398.1  2914.4  395.67  2943.2  396.31  3207.5  394.43  3556.5  393.79
 4355.92388.6243  4434.1   387.5  4471.5  383.98  4472.4  383.18  4480.9  383.18
  4481.9  383.98  4490.9  384.04    4505  387.09  4519.2  388.42  4773.9  390.02
  4795.4  389.44  4816.4  390.86  4858.9  389.22  4936.6  389.45  4950.8  387.66
  4958.2  387.47    4965  388.54  4979.2  386.51  5000.1  386.01  5007.5  387.29
 5032.79388.6245  5050.1  389.59  5170.3  388.96  5269.5   391.1  5324.8  391.02
#Mann= 3 ,-1 , 0
  2632.6      .1       0  4471.5     .07       0  4481.9      .1       0
Bank Sta=4355.92,5032.79
XS Rating Curve= 0 ,0
Exp/Cntr=0.3,0.1

Type RM Length L Ch R = 1 ,35104   ,752,752,752
BEGIN DESCRIPTION:
MACHO CREEK 57.0
END DESCRIPTION:
XS GIS Cut Line= 4
      2087255.56     13455704.02      2087325.01     13453603.35
      2086309.38     13452674.53      2084488.27     13452570.47
#Sta/Elev= 30
    2167  397.24  3106.5  389.22    3877  387.36 4328.02384.9864    4501     385
  4593.5  386.89  4671.2   386.9  4756.3   385.3    4905  387.02  4968.5  385.05
  4982.6  381.79  4984.2  377.35  4985.1  376.55  4994.6  377.35  4996.8  379.42
  5003.6  381.93  5017.8  384.57 5040.33384.9865  5279.9  387.15  5520.4  386.92
  5724.6  388.39  5749.7  387.61  5839.8  389.23    5960  387.95  6050.2  388.81
  6270.5  388.41  6310.6  387.39  6490.9  388.45  6741.3  392.45  7469.2   411.6
#Mann= 3 ,-1 , 0
    2167      .1       0  4984.2     .07       0  4994.6      .1       0
Bank Sta=4328.02,5040.33
XS Rating Curve= 0 ,0
Exp/Cntr=0.3,0.1

Type RM Length L Ch R = 1 ,34352   ,719,719,719
BEGIN DESCRIPTION:
MACHO CREEK 56.0
END DESCRIPTION:
XS GIS Cut Line= 4
      2087435.95     13452763.71      2087147.08      13452534.4
      2086968.38     13452504.62      2086379.29     13452498.67
#Sta/Elev= 30
  4594.4  383.32  4615.6  384.11  4892.8  384.03  4914.8   383.9  4921.6  383.36
    4928  383.71 4940.75 382.192  4942.4  381.96  4950.5  383.28  4956.9  381.15
  4961.4  383.92  4975.5  383.25  4985.3  380.83  4990.3  381.28  4990.5  376.34
  4991.4  375.54    5000  375.54  5000.9  376.34    5016  381.36 5025.33382.1924
  5046.1  383.66  5117.4  384.09  5177.8  383.75  5307.8  384.58  5457.8  384.53
  5577.8  385.96  5657.8  385.98  5697.8  386.82  5707.8  386.37  5733.5   386.6
#Mann= 3 ,-1 , 0
  4594.4      .1       0  4990.5     .07       0  5000.9      .1       0
Bank Sta=4940.75,5025.33
XS Rating Curve= 0 ,0
Exp/Cntr=0.3,0.1

Type RM Length L Ch R = 1 ,33633   ,885,885,885
BEGIN DESCRIPTION:
double MACHO CREEK 55.0
END DESCRIPTION:
XS GIS Cut Line= 3
      2087574.97     13452230.81        2087125.       13451875.
      2086176.04     13452077.13
#Sta/Elev= 30
  4401.6   382.9  4490.8   383.1 4575.81380.2964  4583.3  381.46  4591.4  379.84
  4612.2  379.75  4618.6  382.06  4626.6  380.03    4633  382.08  4641.1  380.51
  4647.5  382.02  4669.3  378.81  4682.7  378.92  4690.8  380.98    4726   381.4
  4740.4  379.43  4761.3  379.65  4775.7  381.93  4804.6   379.6  4833.4  381.13
  4947.2  380.79  4953.6  378.42  4972.1  376.46  4994.8  376.07  4995.7  375.27
  5005.2  376.07  5044.5  378.64 5048.72 380.295  5087.7  381.53  5945.5  384.59
#Mann= 3 ,-1 , 0
  4401.6      .1       0  4994.8     .07       0  5005.2      .1       0
Bank Sta=4575.81,5048.72
XS Rating Curve= 0 ,0
Exp/Cntr=0.3,0.1

Type RM Length L Ch R = 1 ,32748   ,447,447,447
BEGIN DESCRIPTION:
MACHO CREEK 54.0
END DESCRIPTION:
XS GIS Cut Line= 3
       2087084.5     13451444.38      2086780.24     13451464.03
      2085929.96     13451817.97
#Sta/Elev= 30
  4672.2  379.93  4741.8  379.08  4852.1  379.15  4942.3  380.13  4962.3  379.91
  4977.1  378.55 4979.55377.6474  4999.2  371.83  5000.1  371.03  5008.8  371.03
  5009.7  371.83  5014.2  376.44  5017.7377.6491  5026.1  379.29  5048.9  379.48
  5080.3  379.31  5091.1  377.84  5120.5  379.43  5188.6  380.07    5309  380.01
  5351.1   378.4  5356.7   379.1    5386  378.93  5433.6  380.13  5462.9  379.63
  5492.2  380.59    5676  381.88    5723  381.61  5770.7  382.63  5898.1  382.73
#Mann= 3 ,-1 , 0
  4672.2      .1       0  4999.2     .07       0  5009.7      .1       0
Bank Sta=4979.55,5017.7
XS Rating Curve= 0 ,0
Exp/Cntr=0.3,0.1

Type RM Length L Ch R = 1 ,32301   ,377,377,377
BEGIN DESCRIPTION:
MACHO CREEK 53.0
END DESCRIPTION:
XS GIS Cut Line= 3
      2086926.85     13451206.43        2086675.     13451112.18
      2086098.77      13451229.2
#Sta/Elev= 30
  4706.4  379.15  4920.5  378.87  4950.8  377.63  4977.9  377.46 4980.64376.1836
  4985.5  373.92  4990.5  369.35  4991.4  368.55  5000.1  368.55    5001  369.35
  5005.9  371.84  5012.8     377  5017.9   376.8  5026.3  379.04  5097.8   377.9
  5114.1  373.54  5119.2  373.74  5128.4   375.4  5138.5376.1823  5148.8  377.28
    5159  377.54  5164.7  376.21  5169.8  376.21  5179.4  377.39  5189.6  377.84
  5215.3  378.35  5230.4  377.92  5285.8  379.92  5393.7   382.2  5563.3  383.93
#Mann= 4 ,-1 , 0
  4706.4      .1       0  4990.5     .07       0    5001      .1       0
  5285.8     .05       0
Bank Sta=4980.64,5138.5
XS Rating Curve= 0 ,0
Exp/Cntr=0.3,0.1

Type RM Length L Ch R = 1 ,31924   ,311,311,311
BEGIN DESCRIPTION:
MACHO CREEK 52.0
END DESCRIPTION:
XS GIS Cut Line= 5
      2086918.49     13451163.56      2086634.62     13450807.61
      2086359.75     13450857.17      2085895.61     13451132.05
      2085711.03      13451240.1
#Sta/Elev= 30
  4469.7  378.94  4691.8  378.14  4706.2  377.66  4840.7  378.14  4965.2  377.78
  4975.4  377.64  4985.6  376.54 4986.81 375.067  4992.5  368.14  4993.4  367.34
  5002.3  367.34  5003.1  368.14  5005.9  368.96  5016.1  373.84  5036.4  375.39
  5046.3  376.68  5066.9  376.71    5077  374.69 5083.44375.0625  5097.3  376.74
    5105  376.11  5127.8  377.58  5170.1  378.79  5314.4  381.09  5453.9  381.32
  5520.8     382  5563.7  383.05  5593.3  383.02  5651.5  384.23  5957.6  386.21
#Mann= 4 ,-1 , 0
  4469.7      .1       0  4992.5     .07       0  5003.1      .1       0
  5170.1     .05       0
Bank Sta=4986.81,5083.44
XS Rating Curve= 0 ,0
Exp/Cntr=0.3,0.1

Type RM Length L Ch R = 1 ,31613   ,433,433,433
BEGIN DESCRIPTION:
MACHO CREEK 51.0
END DESCRIPTION:
XS GIS Cut Line= 4
      2086960.51     13451166.74      2086706.94     13450830.61
        2086650.       13450650.      2086098.77     13450766.33
#Sta/Elev= 30
  4488.7  378.81  4772.3  377.67  4786.8  375.43  4793.1  376.07  4801.4  374.95
    4816   375.1  4822.2  376.43  4836.8  376.13  4843.1  377.36  4879.2  376.81
  4947.1  377.76  4964.5  376.54  4969.7  377.46 4980.87374.3379    4989  369.94
  4991.5  366.18  4992.4  365.38  5001.3  365.38  5002.1  366.18    5010  373.23
  5020.5  376.87  5248.4   377.6  5298.4  377.01  5329.1  373.12  5337.7  372.87
 5342.35 374.338  5350.6  375.41  5400.6  378.08  5461.9  379.13  5662.5  379.97
#Mann= 4 ,-1 , 0
  4488.7      .1       0  4991.5     .07       0  5002.1      .1       0
  5350.6     .05       0
Bank Sta=4980.87,5342.35
XS Rating Curve= 0 ,0
Exp/Cntr=0.3,0.1

Type RM Length L Ch R = 1 ,31180   ,150,150,150
BEGIN DESCRIPTION:
MACHO CREEK 50.0
END DESCRIPTION:
XS GIS Cut Line= 4
      2088651.27     13450522.32      2087625.22     13450397.32
      2086505.42     13450459.82       2085814.9     13450745.33
#Sta/Elev= 30
  3082.6     387  3260.8   385.8  3421.9  385.02  3572.5  381.88  3924.4  378.96
  3929.4   380.5  3935.1  379.14    4056  377.73  4347.8  377.74  4376.9  376.74
  4717.4  377.29  4937.7  375.05  4947.7  376.05 4969.73373.6737  4991.4  364.62
  4991.9  363.82  5003.7  363.82  5004.2  364.62  5027.9  375.02  5037.9  375.76
  5249.1  376.95  5357.3  376.08  5365.9  375.48  5378.9  370.48  5389.7  370.78
  5397.8373.6747  5411.4  375.09  5471.8  376.46  5955.6  382.02    5985  382.18
#Mann= 7 ,-1 , 0
  3082.6      .1       0  3260.8     .05       0  3421.9      .1       0
  4991.4     .07       0  5004.2      .1       0  5471.8     .05       0
  5955.6      .1       0
Bank Sta=4969.73,5397.8
XS Rating Curve= 0 ,0
Exp/Cntr=0.3,0.1

Type RM Length L Ch R = 1 ,31030   ,494,494,494
BEGIN DESCRIPTION:
MACHO CREEK 49.0
END DESCRIPTION:
XS GIS Cut Line= 3
      2087679.04     13450161.57        2086675.       13450325.
      2085732.44     13450693.25
#Sta/Elev= 30
  3967.5  379.22  4203.1  376.31    4387  376.73  4427.5  375.58    4620   376.8
  4766.9  376.32  4812.5   374.9  4934.1  376.32  4964.5  375.23 4976.26373.0504
  4982.2  370.94  4987.4  370.94  4993.3   364.5  4993.8   363.7  5006.1   364.5
  5006.2  369.26    5017  373.18  5029.5  375.45    5054  374.59  5113.7  376.35
  5231.7  376.47  5325.6  375.55    5331  375.05    5339  371.81  5349.8   371.1
 5357.17373.0484  5371.3  374.67  5444.2  376.32  5849.1  381.08  5996.7  382.35
#Mann= 5 ,-1 , 0
  3967.5      .1       0  4993.3     .07       0  5006.1      .1       0
  5444.2     .05       0  5849.1      .1       0
Bank Sta=4976.26,5357.17
XS Rating Curve= 0 ,0
Exp/Cntr=0.3,0.1

Type RM Length L Ch R = 1 ,30536   ,1308,1308,1308
BEGIN DESCRIPTION:
MACHO CREEK 48.0
END DESCRIPTION:
XS GIS Cut Line= 4
      2087925.01       13449775.      2086575.68     13449919.12
      2086516.65      13449921.2       2084843.3     13450814.42
#Sta/Elev= 30
  3628.1  387.81  4372.3  373.61  4533.2  374.65 4553.19372.1912  4593.6  373.92
  4633.8  370.78    4674  372.96  4694.1  368.75  4734.4  374.21  4834.9  374.88
  4865.1  372.09  4955.6  375.32  4975.7  371.73  4982.9  364.89  4989.4  364.08
  4989.9  363.28  5002.2  364.08  5005.4  368.41  5010.4  366.17  5047.9  369.77
  5057.3  374.89    5063  369.64  5068.7  373.83  5079.2  375.23  5114.1  375.53
 5440.56372.1905  5480.3   373.4  6141.2  382.65  6573.5   385.1    6941  392.34
#Mann= 6 ,-1 , 0
  3628.1      .1       0  4989.4     .07       0  5002.2      .1       0
  5480.3     .05       0  6141.2      .1       0  6573.5     .05       0
Bank Sta=4553.19,5440.56
XS Rating Curve= 0 ,0
Exp/Cntr=0.3,0.1

Type RM Length L Ch R = 1 ,29228   ,814,814,814
BEGIN DESCRIPTION:
MACHO CREEK 47.0
END DESCRIPTION:
XS GIS Cut Line= 3
      2087525.01       13449525.        2086325.       13449425.
      2084826.03     13450579.99
#Sta/Elev= 30
  3777.9  381.57  4322.3  375.43  4359.9  373.85  4400.1  374.49  4490.4  372.16
  4530.5  373.75  4620.8  373.73  4741.2  370.59  4881.7  373.41    4952     372
 4972.09370.1242  4985.2  367.97  4989.2  361.28  4989.7  360.48  5002.1  361.28
  5010.1  362.41  5018.3   367.4  5032.6  372.36  5039.1  373.07  5238.4  374.29
  5395.2  373.05  5474.4  372.22  5502.1  367.56 5513.85 370.127  5560.1  372.48
  5624.4  371.76    5994  379.76  6220.8  380.26  6611.4  384.55  6874.4  390.26
#Mann= 6 ,-1 , 0
  3777.9      .1       0  4989.2     .07       0  5002.1      .1       0
  5395.2     .05       0  6220.8      .1       0  6611.4     .05       0
Bank Sta=4972.09,5513.85
XS Rating Curve= 0 ,0
Exp/Cntr=0.3,0.1

Type RM Length L Ch R = 1 ,28414   ,703,703,703
BEGIN DESCRIPTION:
MACHO CREEK 46.0
END DESCRIPTION:
XS GIS Cut Line= 5
      2086676.53     13449006.88      2086320.65     13449026.41
      2085919.18     13449117.55      2085733.62     13449223.43
       2085361.7     13449600.55
#Sta/Elev= 30
  4176.2  375.39  4661.5  371.29    4777  372.07 4825.19369.1097    4846  366.89
  4876.8   372.3  4952.1  372.21  4983.6  366.77  4988.8  359.94  4989.3  359.14
  5001.2  359.14  5001.7  359.94  5005.3  363.73  5026.9  368.43  5041.2  370.27
  5075.9  371.33    5086  370.71  5107.6  372.25  5121.8  371.96    5145  369.67
  5179.3  366.44  5186.4  367.94  5193.4  365.34  5200.5  365.07  5214.7  366.78
  5221.3369.1087  5313.7  372.13  5490.4   372.8  5525.7  371.42  5687.6  374.34
#Mann= 4 ,-1 , 0
  4176.2      .1       0  4988.8     .07       0  5001.7      .1       0
    5145     .05       0
Bank Sta=4825.19,5221.3
XS Rating Curve= 0 ,0
Exp/Cntr=0.3,0.1

Type RM Length L Ch R = 1 ,27711   ,55,55,55
BEGIN DESCRIPTION:
MACHO CREEK 45.0
END DESCRIPTION:
XS GIS Cut Line= 6
      2086374.93     13448675.28      2085999.91     13448727.36
      2085601.47     13448805.49      2085511.57       13448871.
      2085306.71     13448864.92       2085239.5     13449103.61
#Sta/Elev= 30
  4137.8  373.85  4289.2  372.44  4299.3  370.86  4359.8  370.14 4368.22367.7973
  4392.7  370.34  4562.2  370.86  4623.3  365.27  4664.1  368.96  4687.8   367.3
  4739.3  370.55  4837.1  371.22  4857.7  372.89  4867.9  372.39  4893.6  368.14
  4898.7  368.79  5012.7  363.32  5013.2  362.52  5025.1  362.52  5025.6  363.32
  5032.8  367.62  5066.4  369.75  5071.4  367.33  5074.9 367.798  5100.3  371.15
  5258.8  369.54  5332.1     371  5404.9  370.91  5449.8  369.64  5486.6  370.69
#Mann= 3 ,-1 , 0
  4137.8      .1       0  5012.7     .07       0  5025.6      .1       0
Bank Sta=4368.22,5074.9
XS Rating Curve= 0 ,0
Exp/Cntr=0.3,0.1

Type RM Length L Ch R = 1 ,27656   ,712,712,712
BEGIN DESCRIPTION:
MACHO CREEK 44.0
END DESCRIPTION:
XS GIS Cut Line= 6
      2086364.53     13448604.96      2085755.11     13448683.09
       2085567.3     13448759.72      2085497.85     13448823.61
      2085298.55     13448815.97      2085154.42     13449221.66
#Sta/Elev= 30
  4126.9  373.94  4307.9  371.39 4350.73367.6639  4358.3  366.03  4403.1  370.44
    4449   369.5  4539.8  370.54  4620.4  365.53  4716.6  370.12  4860.2  371.13
    4871  369.76  4889.6  369.99    4895  368.47  4913.6  371.59    4919  367.93
    4925  370.77  4956.7  370.26  4985.1   362.1  4991.9   362.8  4992.8  360.88
  4993.3  360.08  5005.7  360.88  5027.6  364.43 5079.86367.6645  5151.4  370.06
  5268.8  369.61  5350.7  370.95  5468.9  369.27  5518.2   370.8  5668.5  372.07
#Mann= 4 ,-1 , 0
  4126.9      .1       0  4992.8     .07       0  5005.7      .1       0
  5518.2     .05       0
Bank Sta=4350.73,5079.86
XS Rating Curve= 0 ,0
Exp/Cntr=0.3,0.1

Type RM Length L Ch R = 1 ,26944   ,648,648,648
BEGIN DESCRIPTION:
MACHO CREEK 43.0
END DESCRIPTION:
XS GIS Cut Line= 4
      2085697.86      13448667.5      2085396.34     13448367.47
      2085322.99     13448367.47      2082925.02     13449174.99
#Sta/Elev= 30
  4519.1  370.43  4713.8  369.64  4862.3  367.93  4947.6  368.99  4966.1366.0974
  4975.8  364.72  4989.1   358.7  4989.7   357.9  5001.8   357.9  5002.4   358.7
  5005.8  361.01  5017.8  361.64  5023.4  363.66  5028.6  362.39  5047.3  365.65
  5054.8  368.19  5060.1  364.75    5079  366.68  5086.3  366.76  5091.6   365.4
 5099.02366.0984    5174  368.65  5237.3  367.56  5553.5  372.01  5722.7  372.75
  6587.5  380.73    7010  383.69  7217.4  386.35  7284.1  388.07  7548.1  393.25
#Mann= 4 ,-1 , 0
  4519.1      .1       0  4989.1     .07       0  5002.4      .1       0
  7284.1     .05       0
Bank Sta=4966.1,5099.02
XS Rating Curve= 0 ,0
Exp/Cntr=0.3,0.1

Type RM Length L Ch R = 1 ,26296   ,261,261,261
BEGIN DESCRIPTION:
double MACHO CREEK 42.0
END DESCRIPTION:
XS GIS Cut Line= 4
      2085661.07     13448393.47       2085457.1     13447942.12
        2085325.       13447925.      2083724.96     13448725.02
#Sta/Elev= 30
  4310.9  369.45  4625.6  368.52  4671.4  367.47  4682.8  366.03  4700.4  367.66
 4728.53365.1852  4752.1  366.88  4769.8   366.3  4775.2  364.65  4781.1  367.31
  4919.2  365.18  4942.2  362.96  4947.8  359.25  4953.4  360.66  4955.1     357
  4955.7   356.2  4968.4     357  4975.7  360.14  4984.1  357.64  4992.5   358.7
  4998.1  357.87  5014.9  368.17  5221.7  367.98  5252.5   366.9  5274.8  364.54
 5298.81365.1863  5350.3   367.8  5529.2   369.5  5870.2  375.74  6728.3  381.38
#Mann= 3 ,-1 , 0
  4310.9      .1       0  4955.1     .07       0  4968.4      .1       0
Bank Sta=4728.53,5298.81
XS Rating Curve= 0 ,0
Exp/Cntr=0.3,0.1

Type RM Length L Ch R = 1 ,26035   ,228,228,228
BEGIN DESCRIPTION:
MACHO CREEK 41.0
END DESCRIPTION:
XS GIS Cut Line= 5
      2086925.32     13448081.13      2086005.21     13447555.98
      2085536.46     13447573.34      2084677.08      13448011.7
      2083904.55     13448528.18
#Sta/Elev= 30
  3184.5  380.12  3387.4  374.46  3694.2  370.57  3790.7  371.47  3833.9   369.6
  3930.4  369.34  3967.8  370.38  4241.2  366.69  4355.9  368.67  4614.4  368.43
  4862.9  367.05 4958.44364.8107  4968.5  362.49  4984.1  361.82  4996.3  355.93
  4999.4  355.92  5000.4  355.12  5013.7  355.92  5018.6  359.85    5029  362.39
 5071.51364.8104  5168.5  367.88  5264.7  366.15  5296.3  367.08  5332.1  365.06
  5429.7  369.28  5435.3  368.16  5601.5   368.7  6019.8  375.57    6607  379.53
#Mann= 3 ,-1 , 0
  3184.5      .1       0  4999.4     .07       0  5013.7      .1       0
Bank Sta=4958.44,5071.51
XS Rating Curve= 0 ,0
Exp/Cntr=0.3,0.1

Type RM Length L Ch R = 1 ,25807   ,441,441,441
BEGIN DESCRIPTION:
double MACHO CREEK 40.0
END DESCRIPTION:
XS GIS Cut Line= 4
      2085640.41     13447544.66      2085334.42     13447474.87
      2085189.05     13447492.58      2083318.29     13448638.28
#Sta/Elev= 30
  4627.1  367.91  4889.1  366.57 4912.79364.3277  4979.5  359.84  4984.5  361.75
  4993.7  356.59  4994.7  355.79    5008  356.59 5026.18364.3282  5086.9   366.5
  5295.2  367.12    5390  364.83  5420.5  368.06  5426.7  371.42  5432.6  370.99
  5455.7  377.58  5484.8  374.62  5500.2  369.28  5530.8  369.28  5659.5  369.28
  5747.8  369.32  5769.1  371.39  5774.9  374.56  5790.4  374.83  5796.2  377.99
  5827.1  377.63  5842.6   376.3  5848.4  373.67    5891  372.07  7281.1  384.25
#Mann= 5 ,-1 , 0
  4627.1      .1       0  4993.7     .07       0    5008      .1       0
  5530.8     .05       0  5659.5      .1       0
Bank Sta=4912.79,5026.18
XS Rating Curve= 0 ,0
Exp/Cntr=0.3,0.1

Type RM Length L Ch R = 1 ,25366   ,1027,1027,1027
BEGIN DESCRIPTION:
double MACHO CREEK 39.0
END DESCRIPTION:
XS GIS Cut Line= 3
      2085615.68     13447224.24      2085132.44     13447118.51
      2083409.77     13448248.54
#Sta/Elev= 30
  4540.7  366.85  4744.3  366.75 4851.65363.1033  4971.3  362.19  4984.6  356.29
  4985.6  355.49  4998.9  356.29  5012.3  357.47  5031.9  364.82  5059.3  366.15
 5159.37363.1032  5234.1  365.81  5463.1  367.31  5478.2  369.78  5493.3  376.73
    5533  367.67  5565.6   366.6  5601.8  368.91  5622.9  375.58    5644  377.43
  5674.2  376.59  5680.1  373.18  5689.3  373.17  5695.2  369.99  5749.2  369.28
  5797.7  369.44  5818.8  375.05  5839.9  377.43  5891.2  370.63  7095.6  381.12
#Mann= 5 ,-1 , 0
  4540.7      .1       0  4984.6     .07       0  4998.9      .1       0
    5533     .05       0  5749.2      .1       0
Bank Sta=4851.65,5159.37
XS Rating Curve= 0 ,0
Exp/Cntr=0.3,0.1

Type RM Length L Ch R = 1 ,24339   ,488,488,488
BEGIN DESCRIPTION:
double MACHO CREEK 38.0
END DESCRIPTION:
XS GIS Cut Line= 4
      2085437.51     13446705.16       2085095.3     13446672.27
      2084626.03     13446772.06      2083756.78     13447746.03
#Sta/Elev= 30
  4405.1  365.09  4538.2  365.78  4658.8  364.55  4730.9  365.05 4798.79362.4354
  4851.4  361.12  4958.6  360.53  4973.7  357.49  4978.8  358.25  4984.3  355.95
  4997.5  355.31  4998.6  354.51  5010.9  354.51    5012  355.31  5023.3  358.81
  5028.4  356.84  5045.7  358.25  5122.5  358.31  5147.9  359.66  5166.9  359.08
  5172.1  360.06  5178.6  359.18  5238.5  363.76 5272.38362.4354    5302  364.84
  5352.2  364.17    5380  365.38  5578.7  366.13  6152.3  372.64  6534.1  375.57
#Mann= 5 ,-1 , 0
  4405.1      .1       0  4730.9     .12       0  4958.6      .1       0
  4997.5     .07       0    5012      .1       0
Bank Sta=4798.79,5272.38
XS Rating Curve= 0 ,0
Exp/Cntr=0.3,0.1

Type RM Length L Ch R = 1 ,23851   ,546,546,546
BEGIN DESCRIPTION:
double MACHO CREEK 37.0
END DESCRIPTION:
XS GIS Cut Line= 3
      2085047.12     13446421.35        2084825.       13446475.
      2083225.03     13447874.97
#Sta/Elev= 30
  4764.7  364.31  4821.1  364.18    4880  364.27 4908.21362.2564  4922.9  362.04
  4969.7  358.28  4974.8   355.6  4983.4  353.24  4984.5  352.44  4996.8  352.44
  4997.9  353.24    5007  357.43  5021.2  360.04  5049.7  354.81  5057.3  355.81
  5071.5  360.02  5082.2  359.43  5092.4  359.32  5106.6  362.55 5117.23362.2568
  5141.7   364.4  5227.2  364.01  5432.2  365.81  5531.8   364.6  5815.6  368.29
  5829.9  367.69  5843.6   368.5  7048.5  380.44  7097.9  380.18  7119.2  381.25
#Mann= 6 ,-1 , 0
  4764.7      .1       0  4821.1     .12       0  4922.9     .07       0
  4983.4     .07       0  4997.9     .07       0  5082.2      .1       0
Bank Sta=4908.21,5117.23
XS Rating Curve= 0 ,0
Exp/Cntr=0.3,0.1

Type RM Length L Ch R = 1 ,23305   ,583,583,583
BEGIN DESCRIPTION:
double MACHO CREEK 36.0
END DESCRIPTION:
XS GIS Cut Line= 4
      2084936.41     13445978.06       2084656.5     13445972.85
      2084605.47     13446001.04      2083813.71     13447181.08
#Sta/Elev= 30
  4699.7  362.93 4759.86 361.996  4821.1  361.68  4891.1  363.06  4901.1  362.84
  4931.1  358.62  4961.1   360.7  4971.2   358.7  4977.9  353.93  4983.4  353.93
  4989.2  352.35  4990.3  351.55  5002.6  351.55  5003.7  352.35  5012.5   355.3
  5034.3  359.79  5078.2  360.96  5135.3  360.58  5222.3  362.64  5258.3  362.18
  5300.3  360.27  5343.8  360.61  5351.3  361.76  5357.4  360.81  5372.4  360.72
 5444.06361.9966  5480.4   363.5  5849.5  365.74  6092.6  368.88    6459  371.33
#Mann= 3 ,-1 , 0
  4699.7      .1       0  4989.2     .07       0  5003.7      .1       0
Bank Sta=4759.86,5444.06
XS Rating Curve= 0 ,0
Exp/Cntr=0.3,0.1

Type RM Length L Ch R = 1 ,22722   ,685,685,685
BEGIN DESCRIPTION:
double MACHO CREEK 35.0
END DESCRIPTION:
XS GIS Cut Line= 3
      2084834.45     13445611.31        2084325.       13445575.
      2084124.18       13445670.
#Sta/Elev= 30
  4468.9  362.06 4512.28361.7337  4568.6  360.46  4638.8  360.96  4658.8  358.71
  4668.9  360.22    4709  360.13    4719  358.83    4739  360.69  4759.1  361.03
  4799.2  359.61  4819.2  360.15    4896  359.09  4939.5  359.36  4958.7   357.2
  4977.1  354.27  4982.4  354.27  4986.5  352.62  4987.6  351.82  4999.9  351.82
    5001  352.62    5011   356.5  5016.5  357.23  5023.9  360.82 5041.53361.7323
    5046  363.04  5062.1  362.33  5068.1  364.13  5090.3  365.55  5201.8   367.3
#Mann= 5 ,-1 , 0
  4468.9      .1       0    4896     .12       0  4958.7      .1       0
  4986.5     .07       0    5001      .1       0
Bank Sta=4512.28,5041.53
XS Rating Curve= 0 ,0
Exp/Cntr=0.3,0.1

Type RM Length L Ch R = 1 ,22037   ,833,833,833
BEGIN DESCRIPTION:
MACHO CREEK 34.0
END DESCRIPTION:
XS GIS Cut Line= 3
      2084811.44      13445388.8      2084559.71      13445193.5
      2083995.72     13445548.46
#Sta/Elev= 30
  4780.9  361.92 4852.94361.5995  4915.7  361.19  4926.8  358.33  4938.3   355.5
  4944.7  356.54  4952.8  354.16  4959.2  355.62  4966.4   352.4  4967.5   351.6
  4980.9   352.4  5008.9  352.52  5016.9  353.46  5023.4   356.2  5037.9  357.87
  5080.2  356.58    5242  359.01  5247.9  357.74  5257.3   358.8  5263.4  357.73
  5293.8  359.26  5299.7  357.99    5315  360.35  5336.2  360.81  5378.6  361.14
  5400.5  358.66  5409.2  360.16 5481.61361.5993  5697.7  366.77  5765.9  366.77
#Mann= 5 ,-1 , 0
  4780.9      .1       0  4926.8     .12       0  4966.4     .07       0
  4980.9     .12       0  5263.4      .1       0
Bank Sta=4852.94,5481.61
XS Rating Curve= 0 ,0
Exp/Cntr=0.3,0.1

Type RM Length L Ch R = 1 ,21204   ,650,650,650
BEGIN DESCRIPTION:
MACHO CREEK 33.0
END DESCRIPTION:
XS GIS Cut Line= 4
      2084755.02     13444898.36      2084442.52     13444833.26
      2084212.49     13445032.91      2083895.03     13445458.19
#Sta/Elev= 30
  4601.9  358.18    4607  357.59  4612.1   356.4  4622.3   355.8  4699.3  354.44
  4775.6  356.27  4811.9  356.17  4857.3     355  4934.5   355.4  4984.2  351.92
  4985.4  351.12  4997.7  351.12  4998.8  351.92  4999.1  351.92    5020  353.55
  5026.7  357.31  5040.9  360.16  5048.5  360.41  5112.1  359.73  5126.4  360.41
    5133  360.19  5147.3  358.04  5154.9  358.07  5161.5  359.93    5190  357.53
  5218.5  360.45 5386.42361.5511  5446.9  362.37  5482.4  363.76  5756.4   365.8
#Mann= 7 ,-1 , 0
  4601.9      .1       0    4607     .12       0  4699.3      .1       0
  4811.9     .12       0  4984.2     .07       0  4998.8     .12       0
  4999.1      .1       0
Bank Sta=4601.9,5386.42
XS Rating Curve= 0 ,0
Exp/Cntr=0.3,0.1

Type RM Length L Ch R = 1 ,20554   ,78,78,78
BEGIN DESCRIPTION:
MACHO CREEK 32.0
END DESCRIPTION:
XS GIS Cut Line= 6
      2084847.18     13444687.33      2084729.17     13444361.53
      2084568.58     13444322.47      2084416.67     13444348.51
      2084325.52     13444409.27      2083700.79     13445450.49
#Sta/Elev= 30
  4495.8   360.1  4527.9  362.62  4558.1   362.3  4593.8  360.06  4624.4   356.9
  4716.6  354.85  4799.5  353.18  4841.2  353.93  4845.6  353.08  4855.5  353.52
  4880.7     352  4884.8  351.92  4885.9  351.12  4898.2  351.12  4899.4  351.92
  5087.4  351.92  5114.7  352.79  5119.7  351.94  5150.4  353.17  5172.3  353.27
  5187.3  354.39  5208.3  354.06  5273.8  358.76  5346.4  360.08  5564.1  361.39
    5668  360.03  5761.3  360.13 5929.38361.5479  6125.8  363.94  6490.7  366.04
#Mann= 7 ,-1 , 0
  4495.8      .1       0  4716.6     .05       0  4799.5      .1       0
  4880.7     .05       0  4884.8    .033       0  4899.4     .05       0
  5150.4      .1       0
Bank Sta=4495.8,5929.38
XS Rating Curve= 0 ,0
Exp/Cntr=0.3,0.1

Type RM Length L Ch R = 1 ,20476   ,86,86,86
BEGIN DESCRIPTION:
MACHO CREEK 31.0
END DESCRIPTION:
XS GIS Cut Line= 6
      2084893.43     13444514.35      2084837.67     13444400.59
      2084707.46      13444261.7      2084520.83     13444257.36
      2084338.54     13444292.09      2083609.97     13445319.92
#Sta/Elev= 30
    4599  359.43  4627.8  359.41  4650.3  360.49  4655.9  362.32  4678.4   362.8
    4781  361.36  4809.4  362.52  4830.4   361.2  4837.7  362.41  4844.6  361.16
  4851.9  362.53  4858.7  361.25    4866  362.85  4872.9  361.82  4880.2  363.36
    4887  362.49  4908.5  364.09  4978.5  361.56  4999.6  363.15    5115  363.68
    5428  360.62  5432.2  361.72  5462.3  359.02  5463.4  358.22  5476.9  359.02
  5478.1  360.11    5570  361.01  5806.3  359.66 5991.21361.1967  6550.7  365.25
#Mann= 5 ,-1 , 0
    4599      .1       0  4999.6     .05       0    5115      .1       0
  5462.3    .033       0  5476.9      .1       0
Bank Sta=4599,5991.21
XS Rating Curve= 0 ,0
Exp/Cntr=0.3,0.1

Type RM Length L Ch R = 1 ,20390   ,743,743,743
BEGIN DESCRIPTION:
MACHO CREEK 30.0
END DESCRIPTION:
XS GIS Cut Line= 6
      2085038.43     13444476.04      2084941.84     13444400.59
      2084815.97     13444192.26      2084438.37     13444183.58
      2084260.42     13444309.45      2083570.32      13445307.7
#Sta/Elev= 30
    4489  358.44  4641.5   358.7  4671.9  357.84  4677.7     356  4687.4  355.52
  4723.2  358.12  4825.2   356.4 4861.65354.5044  4905.9  350.96    4926  353.48
  4957.2  355.05    4976  350.92    4996  349.06    5026   353.5    5166  358.59
  5293.8  356.25  5359.1  357.55  5365.2  358.68  5472.3  358.71  5573.7  361.33
  5587.3  348.74  5588.5  347.94  5601.9  348.74  5603.3  352.94 5604.72 354.507
  5609.5  359.78  5688.4  360.78  5976.5  359.47  6486.8  364.21  6664.2  364.61
#Mann= 3 ,-1 , 0
    4489      .1       0  5587.3     .07       0  5601.9      .1       0
Bank Sta=4861.65,5604.72
XS Rating Curve= 0 ,0
Exp/Cntr=0.3,0.1

Type RM Length L Ch R = 1 ,19647   ,476,476,476
BEGIN DESCRIPTION:
MACHO CREEK 29.0
END DESCRIPTION:
XS GIS Cut Line= 4
      2085043.25     13443323.25      2084720.96     13443367.61
      2084520.31     13443598.96      2084417.37     13443799.96
#Sta/Elev= 30
  4334.2   356.1  4413.2  355.67  4483.8  354.15  4574.7  355.25  4725.5  353.42
  4768.2  354.03  4789.1  355.84  4839.5  356.29  4860.3  355.83 4910.17352.2912
  4923.9  350.88  4965.8  351.06  4983.3  348.16  4987.2  344.93  4988.8  344.13
  5001.3  344.13  5002.9  344.93  5005.5     346  5011.1  346.74  5017.5  349.49
  5027.7  350.99  5055.5  352.06  5062.4  351.59 5071.01352.2912  5084.9  352.94
  5107.4  352.38  5144.3  355.06  5160.9  357.27  5166.5  356.35  5191.6  357.48
#Mann= 3 ,-1 , 0
  4334.2      .1       0  4987.2     .07       0  5002.9      .1       0
Bank Sta=4910.17,5071.01
XS Rating Curve= 0 ,0
Exp/Cntr=0.3,0.1

Type RM Length L Ch R = 1 ,19171   ,602,602,602
BEGIN DESCRIPTION:
MACHO CREEK 28.0
END DESCRIPTION:
XS GIS Cut Line= 4
      2084674.37     13443152.46      2084347.76     13443191.81
       2084320.5     13443222.29      2084311.95     13443544.51
#Sta/Elev= 30
    4650  354.44  4699.7  354.44  4713.9  353.17    4740  352.21  4750.1  350.93
  4770.2  352.45  4801.1  353.78  4911.3  354.28  4951.5  353.03  4965.2  351.54
    4967350.4657  4971.7  347.66  4982.4  343.71    4984  342.91  4996.5  342.91
  4998.1  343.71  5011.2  348.32  5018.3  349.45  5032.6  349.77  5043.1  349.31
  5052.6  350.88  5062.6   351.6  5092.6  351.41  5112.6  350.17 5142.84350.4656
  5192.6  352.71  5242.7  351.58  5262.7   352.9  5312.7  353.44  5342.2  354.41
#Mann= 3 ,-1 , 0
    4650      .1       0  4982.4     .07       0  4998.1      .1       0
Bank Sta=4967,5142.84
XS Rating Curve= 0 ,0
Exp/Cntr=0.3,0.1

Type RM Length L Ch R = 1 ,18569   ,878,878,878
BEGIN DESCRIPTION:
MACHO CREEK 27.0
END DESCRIPTION:
XS GIS Cut Line= 3
      2084548.65     13442544.68        2083825.       13443025.
      2081789.99     13443911.85
#Sta/Elev= 30
  4120.2  352.52  4196.4  352.58  4259.5  350.95  4352.7  353.48  4605.3  354.37
  4650.4  352.49 4677.57349.0798  4700.7  346.05  4772.7  348.91    4903  349.87
  4945.1  347.13  4975.2  347.25  4991.5   345.6  4994.3  341.29  4996.7  340.49
  5012.1  341.29  5021.2  343.86  5026.6  346.98  5032.4  347.73  5065.1  346.31
 5084.82349.0788  5125.8  351.16  5131.2  352.54  5172.6  353.02  5230.4  356.54
  5370.5  358.36  5650.4  359.82  6005.6  364.68  6699.6  367.11  7208.6   374.9
#Mann= 3 ,-1 , 0
  4120.2      .1       0  4994.3     .07       0  5012.1      .1       0
Bank Sta=4677.57,5084.82
XS Rating Curve= 0 ,0
Exp/Cntr=0.3,0.1

Type RM Length L Ch R = 1 ,17691   ,880,880,880
BEGIN DESCRIPTION:
MACHO CREEK 26.0
END DESCRIPTION:
XS GIS Cut Line= 3
      2084349.03     13442423.13        2083575.       13442625.
        2081575.       13443825.
#Sta/Elev= 30
  4207.9  352.62  4312.3  353.95  4514.7  353.69  4522.1  352.16    4550  350.83
  4595.7  352.17  4636.2  347.88  4697.8  348.12  4747.3  346.68  4868.7  347.74
 4919.56 346.455  4935.5  344.84  4966.5  346.61  4976.8  344.87    4985  339.94
  4988.6  339.39    4991  338.59  5006.4  339.39  5007.8   341.2  5010.7   341.2
  5015.6  346.32 5023.63346.4541  5132.2  353.97  5147.8  352.24  5159.4   355.9
    5175  357.17    5276  359.25  5649.2  362.29  6640.5  366.92  7340.2  379.24
#Mann= 3 ,-1 , 0
  4207.9      .1       0  4988.6     .07       0  5006.4      .1       0
Bank Sta=4919.56,5023.63
XS Rating Curve= 0 ,0
Exp/Cntr=0.3,0.1

Type RM Length L Ch R = 1 ,16811   ,1776,1776,1776
BEGIN DESCRIPTION:
double MACHO CREEK 25.0
END DESCRIPTION:
XS GIS Cut Line= 3
      2084227.51     13442171.39        2083225.       13442425.
      2081625.04       13442625.
#Sta/Elev= 30
  3951.6  352.55  4325.5  351.66  4387.4  350.42 4403.97345.0393  4439.7  341.76
  4516.6  342.16  4548.7  340.57  4551.1  339.77  4566.5  340.57  4593.4  341.35
  4598.6  344.18  4634.5  341.39  4655.6  342.37  4675.5  346.25  4680.6  345.06
  4707.2   347.2  4839.5  344.54  4967.8   344.6  4995.8  342.52 5082.08 345.038
  5116.7  353.79  5136.9  353.21  5146.9   354.5    5157  358.67  5167.1  359.49
    5351  359.88    5419  357.65  5459.3  359.57    5802  362.73  6598.1  381.59
#Mann= 3 ,-1 , 0
  3951.6      .1       0  4548.7     .07       0  4566.5      .1       0
Bank Sta=4403.97,5082.08
XS Rating Curve= 0 ,0
Exp/Cntr=0.3,0.1

Type RM Length L Ch R = 1 ,15035   ,744,744,744
BEGIN DESCRIPTION:
double MACHO CREEK 24.0
END DESCRIPTION:
XS GIS Cut Line= 4
      2084544.34     13441850.22      2084109.27     13441632.53
      2083973.85     13441665.08      2081675.03     13442474.99
#Sta/Elev= 30
  4447.5   352.4    4534  349.89  4556.4  350.21    4562  351.52  4578.7  349.45
    4629   351.9  4645.8  350.63  4852.6  352.08  4897.3  349.13  4914.1  345.97
 4959.34 341.895  4979.5  337.64  4980.9  334.32  4983.3  333.52  4998.8  334.32
    5007   338.2  5020.7  338.06    5031   339.4 5037.05 341.897  5041.2  343.61
  5054.1  344.68  5082.7  343.86    5325  346.57  5448.8  352.36  5973.3   357.3
  6344.4  357.55  6397.4  352.86  6429.2   357.1  6979.6  364.89  7510.6   381.2
#Mann= 3 ,-1 , 0
  4447.5      .1       0  4980.9     .07       0  4998.8      .1       0
Bank Sta=4959.34,5037.05
XS Rating Curve= 0 ,0
Exp/Cntr=0.3,0.1

Type RM Length L Ch R = 1 ,14291   ,1005,1005,1005
BEGIN DESCRIPTION:
MACHO CREEK 23.0
END DESCRIPTION:
XS GIS Cut Line= 3
      2084708.96     13441188.76      2083906.88     13441304.64
      2083158.42     13441661.98
#Sta/Elev= 30
  3965.4  349.93  4100.8  349.15  4255.6  351.23  4444.3  348.28  4636.3  347.01
  4646.4  346.79  4666.6  343.54  4672.5  341.42  4677.6  342.83    4689340.0198
  4742.8  336.58  4785.8  337.35  4800.1  339.74  4822.2  340.72    4933  341.66
  4950.2  339.22  4978.4  337.52  4986.6  332.74  4989.1  331.94  5004.5  332.74
 5015.05340.0175  5032.8  348.21  5040.9  350.35  5046.5  350.23  5063.6   346.5
  5077.1  350.45  5086.3  351.12  5301.6  352.78  5498.2  356.04  5605.2  356.23
#Mann= 3 ,-1 , 0
  3965.4      .1       0  4986.6     .07       0  5004.5      .1       0
Bank Sta=4689,5015.05
XS Rating Curve= 0 ,0
Exp/Cntr=0.3,0.1

Type RM Length L Ch R = 1 ,13286   ,901,901,901
BEGIN DESCRIPTION:
double MACHO CREEK 22.0
END DESCRIPTION:
XS GIS Cut Line= 3
      2084505.27     13441064.63        2083775.       13440875.
      2082474.98       13441075.
#Sta/Elev= 30
  4224.7  348.16  4462.6  349.31  4503.9  343.92  4545.3  342.07  4617.6  348.35
  4718.1  348.64  4751.9  346.51  4772.6  348.69  4813.9  348.96  4839.8  343.26
    4845  345.11  4875.2   339.9  4880.4  341.67 4901.78338.8353  4915.8  334.88
  4920.9  338.39  4927.5  333.78  4939.2  330.34  4941.7  329.54  4957.2  330.34
  4961.5  334.63  4981.7  335.07  5008.3  331.73 5067.36338.8376  5191.7     349
  5232.1  350.09  5602.7  351.74  5697.5  349.48  5734.2  352.38  6294.5  359.47
#Mann= 3 ,-1 , 0
  4224.7      .1       0  4939.2     .07       0  4957.2      .1       0
Bank Sta=4901.78,5067.36
XS Rating Curve= 0 ,0
Exp/Cntr=0.3,0.1

Type RM Length L Ch R = 1 ,12385   ,1299,1299,1299
BEGIN DESCRIPTION:
MACHO CREEK 21.0
END DESCRIPTION:
XS GIS Cut Line= 5
      2084555.14     13440667.89      2083789.55     13440295.52
      2083307.78     13440300.72      2082763.51       13440720.
      2082625.47     13440826.78
#Sta/Elev= 30
  4059.9  346.55  4173.1  347.53  4325.4  346.13  4516.9  348.46  4697.3  343.34
  4714.3  340.02  4719.9  341.57  4727.3  339.49  4742.4  339.97  4749.5  342.29
  4759.4  342.92  4871.8  343.65  4894.1  342.14 4919.01337.8359  4965.8  333.77
  4975.8  329.87  4976.7  328.28  4979.2  327.48  4994.8  328.28  4995.8  331.97
  5005.8   334.2  5025.8  334.61 5052.57337.8353  5065.8  341.02  5115.8  347.82
  5205.8  347.77  5355.8  351.56  5440.9   352.6  5839.5  351.65  6254.6  356.44
#Mann= 3 ,-1 , 0
  4059.9      .1       0  4976.7     .07       0  4994.8      .1       0
Bank Sta=4919.01,5052.57
XS Rating Curve= 0 ,0
Exp/Cntr=0.3,0.1

Type RM Length L Ch R = 1 ,11086   ,715,715,715
BEGIN DESCRIPTION:
double MACHO CREEK 20.0
END DESCRIPTION:
XS GIS Cut Line= 5
      2084415.93     13440267.42      2084363.84     13439913.24
      2084236.56     13439699.12      2083531.94     13439870.36
      2082085.06     13441194.87
#Sta/Elev= 30
  4366.4   346.1  4490.1  345.45  4530.6  342.61  4609.9  342.17  4614.9  340.55
  4679.6  344.14  4724.4  344.17  4772.9  339.38  4815.7  337.51  4831.3  337.34
  4861.9  340.24  4874.1   338.9  4905.4  339.64 4921.51335.5307  4932.6  332.92
  4948.2  331.85  4978.7  331.62  4986.6  328.21  4989.1  327.41  5004.7  328.21
    5006  332.49 5036.48335.5299  5201.5  337.04  5312.8  344.13  5427.9  345.95
  5819.9  347.31  6110.4  351.86  6372.3  350.35    6740  352.88  7660.2  365.83
#Mann= 3 ,-1 , 0
  4366.4      .1       0  4986.6     .07       0  5004.7      .1       0
Bank Sta=4921.51,5036.48
XS Rating Curve= 0 ,0
Exp/Cntr=0.3,0.1

Type RM Length L Ch R = 1 ,10371   ,564,564,564
BEGIN DESCRIPTION:
MACHO CREEK 19.0
END DESCRIPTION:
XS GIS Cut Line= 3
      2084874.99     13439824.99        2084175.       13439125.
        2082575.       13440675.
#Sta/Elev= 30
  4018.8  358.67  4287.5   349.1  4527.9  345.67  4598.6  342.99    4641     339
  4711.8  338.66 4776.16334.8954  4796.6  332.42  4810.7  335.73  4824.9  336.03
  4853.2  330.56  4909.7  329.91    4938  337.72  4966.3  334.11  4980.5  329.94
  4985.5  325.52    4988  324.72  5003.6  325.52  5012.2  325.88  5015.8  329.23
  5022.8  327.59    5030  331.25 5067.54334.8965  5270.5  338.45  5362.3   335.6
  5517.9  345.19  6133.2   347.7  6331.3  350.95  6840.4  351.17  7236.4  356.84
#Mann= 3 ,-1 , 0
  4018.8      .1       0  4985.5     .07       0  5003.6      .1       0
Bank Sta=4776.16,5067.54
XS Rating Curve= 0 ,0
Exp/Cntr=0.3,0.1

Type RM Length L Ch R = 1 ,9807    ,727,727,727
BEGIN DESCRIPTION:
MACHO CREEK 18.0
END DESCRIPTION:
XS GIS Cut Line= 3
        2084975.       13438925.        2084325.       13438675.
      2083144.92     13438803.77
#Sta/Elev= 30
  4307.3  355.83  4382.3  352.71  4491.6  350.68  4564.4   347.9  4600.9  348.38
  4715.5  346.61  4864.4  342.35  4909.4   343.1  4939.4  342.05  4950.1  340.28
  4958.7  335.96 4964.68334.2617  4971.6   331.3  4982.3  330.33    4985  327.45
  4987.5  326.65  5000.7  326.65  5003.2  327.45  5003.7  329.04  5084.2  333.02
  5114.4  333.79  5134.5  332.03  5154.6  332.02 5180.33334.2597  5275.3  338.54
  5345.7  338.47  5627.4   344.3  6019.7  344.27  6120.3  345.25  6190.8   344.6
#Mann= 3 ,-1 , 0
  4307.3      .1       0    4985     .07       0  5003.2      .1       0
Bank Sta=4964.68,5180.33
XS Rating Curve= 0 ,0
Exp/Cntr=0.3,0.1

Type RM Length L Ch R = 1 ,9080    ,784,784,784
BEGIN DESCRIPTION:
MACHO CREEK 17.0
END DESCRIPTION:
XS GIS Cut Line= 4
      2084727.57     13438262.91      2084163.31     13438087.12
      2084009.23     13438308.47      2083520.98     13438577.55
#Sta/Elev= 30
  4341.3  349.13  4691.1  340.71  4718.4  337.66  4756.1  340.17  4878.2  337.34
  4899.1  339.29    4937  339.07  4943.1  338.41 4953.13333.4868  4972.7  326.99
  4984.6  325.48  4987.1  324.68  5002.8  325.48    5015  328.87  5109.8  333.86
  5196.2  333.11  5252.5  330.01  5298.2   332.1  5328.1  328.19  5343.9  328.86
  5349.9  331.85  5355.6  330.65    5366  333.82 5397.16333.4861  5431.3  336.31
  5474.8  336.59  5490.9  339.27  5518.4  338.01  5549.4  341.24  5759.5  343.92
#Mann= 3 ,-1 , 0
  4341.3      .1       0  4984.6     .07       0  5002.8      .1       0
Bank Sta=4953.13,5397.16
XS Rating Curve= 0 ,0
Exp/Cntr=0.3,0.1

Type RM Length L Ch R = 1 ,8296    ,565,565,565
BEGIN DESCRIPTION:
MACHO CREEK 16.0
END DESCRIPTION:
XS GIS Cut Line= 4
      2084716.65     13438082.77       2083952.8     13438000.31
      2083529.63     13438258.56       2083334.3     13438558.06
#Sta/Elev= 30
  3702.6  348.54  4086.5   339.6  4106.6   334.8 4146.64332.4159    4177  333.68
  4198.2  336.52  4207.2  338.79  4227.3  339.75  4267.5  339.68  4368.1  333.66
  4428.4  331.55  4661.9  333.11  4814.9  330.44    4873  331.73  4909.7  328.67
  4966.4  329.65  4988.3  328.25  4990.8  327.45    5004  327.45  5006.5  328.25
 5027.28 332.415  5039.6   335.6    5046  340.48  5054.7  342.47  5069.8  343.38
  5096.9  342.52  5105.7  343.23    5118  342.25  5148.2  343.56  5324.2  343.67
#Mann= 3 ,-1 , 0
  3702.6      .1       0  4988.3     .07       0  5006.5      .1       0
Bank Sta=4146.64,5027.28
XS Rating Curve= 0 ,0
Exp/Cntr=0.3,0.1

Type RM Length L Ch R = 1 ,7731    ,815,815,815
BEGIN DESCRIPTION:
MACHO CREEK 15.0
END DESCRIPTION:
XS GIS Cut Line= 4
      2084744.92     13438019.84      2083752.25     13437831.47
      2083633.79     13437781.13      2083289.35     13437915.44
#Sta/Elev= 30
  3939.8  348.53  4306.1  340.22  4317.9  338.41  4346.9  336.47  4365.1   332.7
 4403.78330.7404  4428.3  329.71  4438.5   332.6  4474.7  338.02  4519.9  340.16
  4611.5  332.22  4672.6  330.31  4774.4  331.22  4886.3  328.67    4903  328.95
  4916.9  330.82  4968.9  331.16  4982.4  329.03  4990.7  326.15  4991.5  323.41
    4994  322.61  5009.7  323.41  5012.4  326.67  5105.1330.7395  5128.4  334.68
  5133.7  334.62    5142  338.38  5163.6  342.68  5375.7  340.53  5448.6  340.82
#Mann= 3 ,-1 , 0
  3939.8      .1       0  4991.5     .07       0  5009.7      .1       0
Bank Sta=4403.78,5105.1
XS Rating Curve= 0 ,0
Exp/Cntr=0.3,0.1

Type RM Length L Ch R = 1 ,6916    ,541,541,541
BEGIN DESCRIPTION:
MACHO CREEK 14.0
END DESCRIPTION:
XS GIS Cut Line= 4
      2084799.16     13437913.51      2084332.58     13437789.81
      2084204.54     13437555.43      2083692.37     13437440.41
#Sta/Elev= 30
  4437.1  348.59  4564.1  345.46  4751.8  343.25  4865.6  339.88  4880.6  337.58
  4886.3  334.03  4896.6  331.82    4907   330.3  4915.6  332.43  4919.4  328.96
  4928.1  330.03 4932.77328.7757  4949.9  326.33  4971.7  325.05  4982.2   323.2
  4984.6  320.42  4987.1  319.62  5000.3  319.62  5002.8  320.42    5004  323.94
  5016.4  327.04  5039.2  329.41 5216.55328.7765  5247.9   329.4  5260.3  330.91
    5352  330.82  5395.4  332.91  5438.7  336.06    5482   337.7  5711.8  340.14
#Mann= 3 ,-1 , 0
  4437.1      .1       0  4984.6     .07       0  5002.8      .1       0
Bank Sta=4932.77,5216.55
XS Rating Curve= 0 ,0
Exp/Cntr=0.3,0.1

Type RM Length L Ch R = 1 ,6375    ,607,607,607
BEGIN DESCRIPTION:
double MACHO CREEK 13.0
END DESCRIPTION:
XS GIS Cut Line= 3
      2084975.03     13437825.02      2084451.94     13437399.18
      2083770.53     13437355.78
#Sta/Elev= 30
  4286.6  350.08  4813.1  341.99  4827.4  336.55  4833.9  341.18  4848.2  335.21
  4854.7  338.82  4862.6  334.68  4869.1  338.42    4877  332.82  4883.4  334.14
  4891.3  329.98  4897.8  334.37 4909.62 328.087  4918.6  329.78  4926.5  327.19
    4933  331.27  4940.9  327.25  4947.3  333.19  4955.3  327.54  4960.5  330.64
    4989  319.32  4991.5  318.52  5007.2  319.32  5028.2  324.74  5088.3  323.97
  5104.4  326.37 5234.64328.0876  5328.8  330.11    5429  337.51  5643.9  338.22
#Mann= 3 ,-1 , 0
  4286.6      .1       0    4989     .07       0  5007.2      .1       0
Bank Sta=4909.62,5234.64
XS Rating Curve= 0 ,0
Exp/Cntr=0.3,0.1

Type RM Length L Ch R = 1 ,5768    ,581,581,581
BEGIN DESCRIPTION:
double MACHO CREEK 12.0
END DESCRIPTION:
XS GIS Cut Line= 3
      2085024.97       13436875.        2084275.       13436875.
      2083754.17     13437002.58
#Sta/Elev= 30
  4246.5  348.84  4356.5     345  4626.5  341.23  4736.5  339.06  4766.5  338.05
  4816.5  334.88  4846.5  334.89  4866.5   333.6  4896.5  333.87  4926.5  335.98
  4946.5   336.1  4956.5  332.54 4964.81327.3712  4966.5  326.32  4976.5  323.21
  4996.5  321.88  4997.7  321.31  5000.2  320.51  5013.4  320.51  5015.9  321.31
  5019.8  323.44  5130.3  325.12 5189.66 327.374  5222.7  331.59  5227.9  330.63
  5264.2  335.15  5316.2   335.4  5418.6  337.03  5449.5  336.58  5532.7  337.02
#Mann= 3 ,-1 , 0
  4246.5      .1       0  4997.7     .07       0  5015.9      .1       0
Bank Sta=4964.81,5189.66
XS Rating Curve= 0 ,0
Exp/Cntr=0.3,0.1

Type RM Length L Ch R = 1 ,5187    ,493,493,493
BEGIN DESCRIPTION:
double MACHO CREEK 11.0
END DESCRIPTION:
XS GIS Cut Line= 3
      2085317.38     13436771.74       2084067.4     13436421.74
      2083869.41     13436559.41
#Sta/Elev= 30
  3691.6  356.25  3714.8  356.29    3919  348.46  4078.3  345.02  4119.8  342.47
  4144.4  343.54    4151  342.91  4265.2  341.41  4590.2  339.81  4711.8  335.82
  4784.5  334.59  4918.1  337.08  4929.8  336.52  4940.2  332.28 4948.61326.5468
  4957.4  321.65  4962.6   323.8  4971.4  321.56  4992.3  318.54  4994.8  317.74
    5008  317.74  5010.5  318.54  5022.3  321.45  5043.3  323.31  5058.1  325.61
 5099.07326.5496  5114.8  329.29  5150.9  333.93  5187.5  335.79  5230.8  336.64
#Mann= 3 ,-1 , 0
  3691.6      .1       0  4992.3     .07       0  5010.5      .1       0
Bank Sta=4948.61,5099.07
XS Rating Curve= 0 ,0
Exp/Cntr=0.3,0.1

Type RM Length L Ch R = 1 ,4694    ,471,471,471
BEGIN DESCRIPTION:
double MACHO CREEK 10.0
END DESCRIPTION:
XS GIS Cut Line= 4
      2085224.99       13436175.      2083963.43     13435953.45
      2083781.14     13436036.78      2083846.25      13436487.3
#Sta/Elev= 30
  3605.1  347.63  3899.5  339.37  4329.4  336.36  4497.3  338.78  4610.2  336.29
  4640.7  330.02    4661  331.68  4675.4  335.67  4691.5  333.57  4711.8   335.2
  4721.9  331.29  4729.7  332.26  4734.8  334.87  4752.4  335.22  4782.8  330.51
  4803.2  332.12  4813.3  330.08  4853.9  335.15  4874.2  335.68  4961.2  331.86
 4979.44325.6804    4996  318.33  4998.5  317.53  5014.3  318.33  5067.9  324.68
  5104.8  323.74 5150.54325.6786  5276.6  333.37  5367.5  332.84  5541.6  336.35
#Mann= 3 ,-1 , 0
  3605.1      .1       0    4996     .07       0  5014.3      .1       0
Bank Sta=4979.44,5150.54
XS Rating Curve= 0 ,0
Exp/Cntr=0.3,0.1

Type RM Length L Ch R = 1 ,4223    ,242,242,242
BEGIN DESCRIPTION:
MACHO CREEK 9.0
END DESCRIPTION:
XS GIS Cut Line= 5
      2084275.41      13435555.1      2083751.67     13435633.66
      2083411.35     13435762.47      2082990.34     13435860.56
      2082706.05     13436050.93
#Sta/Elev= 30
  4198.9  341.11  4219.5  341.43  4228.3  340.54  4239.8  337.19  4249.9   336.4
  4504.7  337.49  4603.8  334.71  4637.8   336.9  4674.6  336.37  4773.9  331.61
  4874.6  331.18 4948.08324.9171  4974.3  319.64  4981.6  317.17  4983.1  315.04
  4985.6  314.24  5001.4  315.04  5004.5  317.94  5013.6  321.11  5029.3  322.96
    5035   320.8  5045.7  322.99 5049.49324.9166  5067.1  333.16  5084.3  338.54
  5125.1  341.12  5390.8  347.21  5475.9  351.72  5567.2  352.21  5866.8  362.01
#Mann= 3 ,-1 , 0
  4198.9      .1       0  4983.1     .07       0  5001.4      .1       0
Bank Sta=4948.08,5049.49
XS Rating Curve= 0 ,0
Exp/Cntr=0.3,0.1
