--- PANTHER Cr.prj (project) ---

Proj Title=PANTHER Cr Base Level Engineering
Current Plan=p01
Default Exp/Contr=0.3,0.1
English Units
Geom File=g01
Flow File=f01
Plan File=p01
BEGIN DESCRIPTION:
PANTHER Cr
END DESCRIPTION:

--- PANTHER Cr.p01 (plan) ---

Plan Title=Multiple Run
Short Identifier=Multiple
Geom File=g01
Flow File=f01
Subcritical Flow
K Sum by GR= 0
Std Step Tol= 0.01
Critical Tol= 0.01
Num of Std Step Trials= 20
Max Error Tol= 0.3
Flow Tol Ratio= 0.001
Split Flow NTrial= 30
Split Flow Tol= 0.02
Split Flow Ratio= 0.02
Log Output Level= 0
Friction Slope Method= 1
Unsteady Friction Slope Method= 2
Unsteady Bridges Friction Slope Method= 1
Parabolic Critical Depth
Global Vel Dist=  1 , 1 , 1
Global Log Level= 0
CheckData=True
Encroach Param= -1, 0, 0, 0
BEGIN DESCRIPTION:
Multiple Run
END DESCRIPTION:

--- PANTHER Cr.f01 (steady flow) ---

Flow Title=Multiple
Number of Profiles=7
Profile Names=10-year,25-year,50-year,1pct_min,100-year,1pct_plu,500-year
River Rch & RM= PANTHER Cr,Reach-1,16869
     140     187     225     135     269     537     391
River Rch & RM= PANTHER Cr,Reach-1,14159
     237     326     400     244     487     973     735
River Rch & RM= PANTHER Cr,Reach-1,11339
     346     484     600     370     739    1474    1138
River Rch & RM= PANTHER Cr,Reach-1,5031
     651     940    1189     748    1493    2978    2389
Boundary for River Rch & Prof#=PANTHER Cr,Reach-1,1
Up Type=0
Dn Type=3
Dn Slope=0.005
Boundary for River Rch & Prof#=PANTHER Cr,Reach-1,2
Up Type=0
Dn Type=3
Dn Slope=0.005
Boundary for River Rch & Prof#=PANTHER Cr,Reach-1,3
Up Type=0
Dn Type=3
Dn Slope=0.005
Boundary for River Rch & Prof#=PANTHER Cr,Reach-1,4
Up Type=0
Dn Type=3
Dn Slope=0.005
Boundary for River Rch & Prof#=PANTHER Cr,Reach-1,5
Up Type=0
Dn Type=3
Dn Slope=0.005
Boundary for River Rch & Prof#=PANTHER Cr,Reach-1,6
Up Type=0
Dn Type=3
Dn Slope=0.005
Boundary for River Rch & Prof#=PANTHER Cr,Reach-1,7
Up Type=0
Dn Type=3
Dn Slope=0.005

--- PANTHER Cr.g01 (geometry) ---

Geom Title=Existing Conditions

River Reach=PANTHER Cr,Reach-1
Reach XY= 30
      2056604.36     13520926.21      2055994.46     13520322.04
      2055546.54     13520476.21      2055376.76     13520940.88
      2055027.80     13521229.94      2054265.14     13520702.46
      2053540.80     13520504.54      2052740.80     13520544.54
      2052290.80     13520044.54      2051832.38     13519759.69
      2051755.34     13519234.52      2051510.80     13518934.54
      2051230.80     13518824.54      2050970.80     13518204.54
      2050340.80     13517574.54      2049790.80     13517244.54
      2049340.80     13517214.54      2049156.60     13517037.25
      2048344.97     13516896.20      2047830.80     13516374.54
      2047390.80     13516264.54      2047350.80     13515814.54
      2047500.80     13515364.54      2047240.80     13514644.54
      2047220.80     13514204.54      2046950.80     13513744.54
      2046860.80     13513264.54      2046620.80     13513024.54
      2046210.80     13512854.54      2046140.80     13512704.54

Type RM Length L Ch R = 1,16869,220,220,220
BEGIN DESCRIPTION:
PANTHER Cr 29.0
END DESCRIPTION:
XS GIS Cut Line= 3
      2057236.42     13520219.06      2056481.44     13520823.60
      2056316.34     13521590.33
#Sta/Elev= 30
  4032.8  561.85  4093.6  559.83  4137.1  557.84  4173.7  557.61  4194.5  556.98
  4208.9  555.57  4223.3  555.62  4229.7  555.26  4237.7  556.46  4244.1  555.78
  4258.6  555.97  4265.2  554.73  4273.0  554.30  4308.2  553.44  4316.2  552.89
  4756.3  542.46  4849.2  538.94  4898.8  538.05  4994.1  535.45  4994.6  534.65
  4999.6  534.65  5000.1  535.45  5062.8  537.49  5154.9  538.90  5248.2  539.42
  5472.0  539.66  5543.6  538.81  5573.0  539.31  5645.9  538.79  5784.3  538.69
#Mann=4,-1,0
  4032.8     0.1       0  4093.6    0.05       0  4994.1    0.03       0
  5000.1    0.05       0
Bank Sta=4994.1,5000.1
Exp/Cntr=0.3,0.1

Type RM Length L Ch R = 1,16649,297,297,297
BEGIN DESCRIPTION:
Mapping XS ea9a2835
END DESCRIPTION:
XS GIS Cut Line= 4
      2056824.59     13520241.28      2056561.58     13520342.84
      2056251.68     13520767.32      2056290.60     13521000.80
#Sta/Elev= 30
  4313.1  550.87  4387.6  549.05  4447.5  547.01  4516.3  545.48  4556.6  544.13
  4580.6  543.88  4591.1  543.09  4622.5  542.19  4630.1  542.35  4636.3  541.91
  4644.8  542.03  4715.9  540.52  4736.7  539.74  4780.8  539.07  4786.9  538.57
  4801.6  538.14  4816.3  538.17  4837.1  537.41  4851.8  537.52  4887.3  536.83
  4916.7  536.78  4990.9  534.74  4991.4  533.94  4996.4  533.94  4996.9  534.74
  5052.6  536.33  5167.5  538.20  5233.4  538.28  5289.2  538.92  5357.3  539.08
#Mann=3,-1,0
  4313.1    0.05       0  4990.9    0.03       0  4996.9    0.05       0
Bank Sta=4990.9,4996.9
Exp/Cntr=0.3,0.1

Type RM Length L Ch R = 1,16352,196,196,196
BEGIN DESCRIPTION:
Mapping XS 05213f9e
END DESCRIPTION:
XS GIS Cut Line= 4
      2056655.32     13520082.43      2056420.95     13520126.70
      2056051.16     13520545.97      2056170.48     13520955.79
#Sta/Elev= 30
  4319.3  549.43  4340.0  548.67  4441.7  546.69  4519.9  544.51  4557.8  543.88
  4568.3  543.36  4617.6  542.20  4624.3  541.83  4646.1  541.59  4730.6  539.32
  4738.1  539.45  4744.8  539.05  4836.8  536.72  4844.4  536.71  4865.3  535.90
  4922.2  534.80  4964.8  534.63  4997.0  533.77  4997.5  532.97  5002.5  532.97
  5003.0  533.77  5063.5  535.69  5092.0  536.05  5136.7  535.86  5183.9  536.58
  5261.7  536.91  5361.9  537.91  5417.9  538.09  5467.6  538.89  5543.7  539.08
#Mann=3,-1,0
  4319.3    0.05       0  4997.0    0.03       0  5003.0    0.05       0
Bank Sta=4997,5003
Exp/Cntr=0.3,0.1

Type RM Length L Ch R = 1,16156,327,327,327
BEGIN DESCRIPTION:
Mapping XS 6298171f
END DESCRIPTION:
XS GIS Cut Line= 4
      2056355.89     13519876.68      2056087.62     13519978.26
      2055952.20     13520519.93      2056069.38     13520824.57
#Sta/Elev= 30
  4357.3  544.87  4433.1  542.44  4505.2  540.83  4510.6  541.04  4620.5  539.15
  4682.0  538.68  4702.6  538.98  4717.5  538.68  4723.3  538.29  4743.9  538.10
  4758.7  537.36  4816.0  535.93  4857.3  535.63  4877.2  535.07  4959.7  534.57
  4997.9  533.08  4998.4  532.28  5003.4  532.28  5003.9  533.08  5042.2  534.11
  5047.3  533.88  5083.4  534.80  5088.5  534.60  5165.8  535.47  5224.1  535.43
  5333.4  536.73  5393.4  536.93  5432.9  537.54  5508.0  537.75  5528.9  538.10
#Mann=3,-1,0
  4357.3    0.05       0  4997.9    0.03       0  5003.9    0.05       0
Bank Sta=4997.9,5003.9
Exp/Cntr=0.3,0.1

Type RM Length L Ch R = 1,15829,337,337,337
BEGIN DESCRIPTION:
Mapping XS fd65fa3d
END DESCRIPTION:
XS GIS Cut Line= 4
      2055801.18     13519897.51      2055681.37     13520072.01
      2055686.58     13520585.03      2055961.30     13520828.65
#Sta/Elev= 30
  4485.9  538.02  4531.4  537.32  4554.1  537.77  4567.8  537.77  4596.0  537.21
  4610.9  536.21  4617.0  536.11  4646.8  536.11  4696.3  535.33  4720.6  535.37
  4770.6  534.63  4840.6  534.11  4900.6  532.89  4920.6  533.08  4950.6  532.90
  4960.6  532.58  4997.6  532.21  4998.1  531.41  5003.1  531.41  5003.6  532.21
  5060.6  533.14  5090.6  532.98  5140.6  533.39  5180.6  533.32  5237.5  533.78
  5259.3  534.18  5358.0  535.06  5408.2  535.77  5422.4  535.75  5577.8  538.02
#Mann=3,-1,0
  4485.9    0.05       0  4997.6    0.03       0  5003.6    0.05       0
Bank Sta=4997.6,5003.6
Exp/Cntr=0.3,0.1

Type RM Length L Ch R = 1,15492,584,584,584
BEGIN DESCRIPTION:
Mapping XS 789be39b
END DESCRIPTION:
XS GIS Cut Line= 4
      2055429.12     13520167.87      2055328.43     13520407.43
      2055529.82     13520728.61      2055713.86     13520846.66
#Sta/Elev= 30
  4498.1  532.95  4516.4  532.91  4574.8  531.99  4636.0  531.38  4668.5  531.36
  4696.0  530.91  4696.5  530.11  4701.5  530.11  4702.0  530.91  4722.7  531.09
  4733.6  531.40  4790.5  531.71  4897.7  531.56  4920.3  531.34  4934.2  531.59
  4955.8  531.43  4979.4  531.62  4991.9  531.38  5080.3  531.49  5167.0  532.24
  5180.7  532.14  5211.1  532.72  5226.3  532.93  5232.3  532.75  5253.4  533.28
  5262.0  533.26  5283.8  533.67  5289.8  533.54  5297.7  533.83  5355.7  534.57
#Mann=3,-1,0
  4498.1    0.05       0  4696.0    0.03       0  4702.0    0.05       0
Bank Sta=4696,4702
Exp/Cntr=0.3,0.1

Type RM Length L Ch R = 1,14908,143,143,143
BEGIN DESCRIPTION:
Mapping XS 17d2cd71
END DESCRIPTION:
XS GIS Cut Line= 4
      2055262.46     13520317.14      2055193.02     13520429.99
      2055215.30     13521328.90      2055533.70     13521650.58
#Sta/Elev= 30
  4187.8  531.50  4325.3  530.82  4505.4  531.22  4601.2  530.24  4606.2  530.54
  4705.4  529.75  4845.5  529.81  4895.5  529.41  4945.5  529.50  5003.0  528.94
  5220.6  528.38  5221.1  527.58  5226.1  527.58  5226.6  528.38  5273.1  528.70
  5280.2  528.52  5287.2  528.83  5308.5  528.83  5322.6  529.15  5336.7  528.90
  5343.8  529.27  5379.2  529.17  5386.2  529.54  5435.7  529.35  5485.2  529.76
  5492.3  529.49  5598.3  530.08  5619.6  529.85  5640.8  530.05  5672.1  529.68
#Mann=3,-1,0
  4187.8    0.05       0  5220.6    0.03       0  5226.6    0.05       0
Bank Sta=5220.6,5226.6
Exp/Cntr=0.3,0.1

Type RM Length L Ch R = 1,14765,258,258,258
BEGIN DESCRIPTION:
Mapping XS 57017fa9
END DESCRIPTION:
XS GIS Cut Line= 4
      2055048.93     13520305.03      2055120.10     13520520.27
      2055124.16     13521646.61      2054958.53     13521754.28
#Sta/Elev= 30
  4078.7  527.42  4114.7  527.31  4141.2  527.80  4172.9  530.30  4184.0  529.70
  4226.1  529.40  4310.3  530.66  4400.1  530.96  4560.1  530.26  4580.1  529.43
  4660.1  527.82  4680.1  528.09  4720.1  527.57  4750.1  528.10  4820.1  528.40
  4900.1  527.47  4920.1  527.63  4970.1  526.80  5097.1  526.22  5097.6  525.42
  5102.6  525.42  5103.1  526.22  5180.1  526.31  5200.1  526.88  5240.1  527.09
  5280.1  526.83  5420.1  529.97  5466.5  529.68  5567.2  530.20  5629.3  529.95
#Mann=3,-1,0
  4078.7    0.05       0  5097.1    0.03       0  5103.1    0.05       0
Bank Sta=5097.1,5103.1
Exp/Cntr=0.3,0.1

Type RM Length L Ch R = 1,14507,348,348,348
BEGIN DESCRIPTION:
Mapping XS ef49a1f4
END DESCRIPTION:
XS GIS Cut Line= 4
      2054963.86     13520471.70      2054993.36     13520676.52
      2054948.23     13521011.59      2054804.11     13521376.22
#Sta/Elev= 30
  4330.5  529.46  4354.0  530.17  4364.1  530.07  4371.4  529.45  4376.4  528.75
  4384.3  528.19  4404.6  529.12  4441.8  529.34  4446.9  529.71  4537.4  529.62
  4634.6  528.47  4677.2  527.74  4778.1  525.26  4808.3  525.80  4868.9  525.35
  4896.6  525.74  4921.0  525.33  4986.7  524.75  4997.5  524.83  5026.1  523.71
  5026.6  522.91  5031.6  522.91  5032.1  523.71  5051.2  524.20  5083.2  525.56
  5088.6  526.10  5094.2  526.34  5137.3  526.78  5202.2  527.88  5267.6  528.21
#Mann=3,-1,0
  4330.5    0.05       0  5026.1    0.03       0  5032.1    0.05       0
Bank Sta=5026.1,5032.1
Exp/Cntr=0.3,0.1

Type RM Length L Ch R = 1,14159,231,231,231
BEGIN DESCRIPTION:
Mapping XS cefee682
END DESCRIPTION:
XS GIS Cut Line= 4
      2054966.50     13520294.58      2054784.86     13520381.36
      2054528.59     13521293.46      2054560.45     13521404.97
#Sta/Elev= 30
  4255.0  526.93  4355.6  526.12  4383.8  526.79  4406.5  526.21  4429.2  526.11
  4451.9  526.24  4509.0  527.53  4615.9  528.17  4688.6  527.58  4734.2  526.80
  4813.2  524.63  4846.8  524.02  4875.6  523.97  4880.8  523.38  4896.3  523.06
  4937.9  523.61  4976.4  522.77  4976.9  521.97  4981.9  521.97  4982.4  522.77
  4993.4  523.14  5010.6  522.89  5027.5  523.24  5041.8  522.89  5072.9  523.80
  5106.0  524.05  5187.2  526.24  5247.5  527.08  5320.8  527.57  5519.7  527.59
#Mann=3,-1,0
  4255.0    0.05       0  4976.4    0.03       0  4982.4    0.05       0
Bank Sta=4976.4,4982.4
Exp/Cntr=0.3,0.1

Type RM Length L Ch R = 1,13928,239,239,239
BEGIN DESCRIPTION:
Mapping XS de16e401
END DESCRIPTION:
XS GIS Cut Line= 4
      2054710.17     13520266.34      2054597.20     13520272.39
      2054308.63     13521226.87      2054349.00     13521354.03
#Sta/Elev= 30
  4346.0  524.89  4401.2  524.48  4451.3  524.33  4518.9  524.46  4629.0  526.44
  4681.2  526.70  4733.5  526.67  4858.8  524.43  4935.2  522.20  4952.9  522.33
  4968.2  521.87  5006.3  521.41  5015.6  521.94  5034.1  522.17  5057.3  522.07
  5088.7  522.26  5105.2  521.94  5116.9  521.17  5117.4  520.37  5122.6  520.37
  5123.1  521.17  5171.1  523.24  5176.3  523.25  5209.2  524.55  5242.2  525.22
  5313.3  525.94  5391.6  526.28  5417.4  526.01  5497.7  526.25  5589.7  526.09
#Mann=3,-1,0
  4346.0    0.05       0  5116.9    0.03       0  5123.1    0.05       0
Bank Sta=5116.9,5123.1
Exp/Cntr=0.3,0.1

Type RM Length L Ch R = 1,13689,164,164,164
BEGIN DESCRIPTION:
Mapping XS 8c028327
END DESCRIPTION:
XS GIS Cut Line= 4
      2054518.49     13520169.48      2054342.94     13520262.30
      2054114.91     13521121.93      2054150.61     13521217.12
#Sta/Elev= 30
  4353.3  525.64  4425.1  524.28  4485.0  523.42  4561.6  523.24  4585.7  522.94
  4601.8  523.32  4642.0  523.57  4717.2  524.84  4757.4  524.95  4813.3  524.40
  4947.8  521.52  4978.8  520.45  4988.2  519.60  4990.3  519.12  4990.8  518.32
  4996.0  518.32  4996.5  519.12  4999.5  519.75  5009.9  520.47  5051.3  519.98
  5092.7  520.30  5113.9  520.05  5143.8  521.07  5189.2  521.84  5264.4  523.63
  5309.9  524.29  5379.8  524.72  5425.1  524.60  5497.9  524.92  5542.9  524.87
#Mann=3,-1,0
  4353.3    0.05       0  4990.3    0.03       0  4996.5    0.05       0
Bank Sta=4990.3,4996.5
Exp/Cntr=0.3,0.1

Type RM Length L Ch R = 1,13525,406,406,406
BEGIN DESCRIPTION:
Mapping XS 951a4a6d
END DESCRIPTION:
XS GIS Cut Line= 4
      2054328.81     13520167.46      2054153.25     13520173.51
      2053997.87     13521071.49      2054063.91     13521271.60
#Sta/Elev= 30
  4336.1  523.43  4553.9  522.04  4574.2  522.23  4604.6  522.00  4763.7  523.02
  4888.8  520.48  4970.0  519.93  4980.1  519.51  4990.3  519.68  4997.7  518.28
  5002.8  518.51  5007.4  518.23  5007.9  517.43  5013.1  517.43  5013.6  518.23
  5020.7  519.20  5030.8  519.40  5062.5  519.21  5101.9  519.46  5112.0  519.14
  5122.3  519.27  5231.7  522.33  5315.0  523.50  5494.5  523.84  5552.7  523.49
  5558.0  523.68  5584.4  523.45  5589.7  523.65  5616.2  523.32  5633.8  523.44
#Mann=3,-1,0
  4336.1    0.05       0  5007.4    0.03       0  5013.6    0.05       0
Bank Sta=5007.4,5013.6
Exp/Cntr=0.3,0.1

Type RM Length L Ch R = 1,13119,798,798,798
BEGIN DESCRIPTION:
Mapping XS 690ba5f7
END DESCRIPTION:
XS GIS Cut Line= 4
      2054068.01     13520192.15      2053753.78     13520245.97
      2053633.99     13520739.02      2053919.80     13520990.19
#Sta/Elev= 30
  4382.2  521.63  4527.3  520.76  4567.9  519.84  4598.3  519.90  4649.0  519.38
  4665.0  519.41  4670.0  519.89  4703.1  519.78  4716.2  520.04  4846.7  519.58
  4925.0  518.25  4966.8  518.03  4971.9  517.91  4977.9  517.15  5013.7  516.97
  5015.9  516.36  5016.4  515.56  5021.6  515.56  5022.1  516.36  5055.5  517.57
  5080.8  517.50  5091.1  517.08  5102.4  517.30  5139.0  519.07  5180.7  520.19
  5235.0  521.07  5305.2  521.62  5362.1  521.39  5447.5  522.52  5588.9  523.09
#Mann=3,-1,0
  4382.2    0.05       0  5015.9    0.03       0  5022.1    0.05       0
Bank Sta=5015.9,5022.1
Exp/Cntr=0.3,0.1

Type RM Length L Ch R = 1,12321,225,225,225
BEGIN DESCRIPTION:
Mapping XS 5369a172
END DESCRIPTION:
XS GIS Cut Line= 4
      2053059.33     13520141.81      2052892.67     13520291.11
      2052936.07     13520803.26      2053114.75     13520980.20
#Sta/Elev= 30
  4480.5  518.02  4584.8  519.76  4648.4  519.64  4787.2  516.82  4792.3  517.01
  4906.7  514.25  4979.1  513.65  4986.0  512.88  4986.5  512.08  4991.9  512.08
  4992.4  512.88  5019.3  513.60  5069.4  515.79  5099.6  515.02  5129.7  515.21
  5216.6  517.69  5261.1  517.68  5303.5  518.76  5310.6  518.54  5317.7  518.92
  5367.2  519.38  5388.4  520.09  5395.5  519.91  5402.5  520.41  5423.8  520.55
  5430.8  521.07  5437.9  520.82  5459.1  521.56  5466.2  521.44  5469.7  521.93
#Mann=3,-1,0
  4480.5    0.05       0  4986.0    0.03       0  4992.4    0.05       0
Bank Sta=4986,4992.4
Exp/Cntr=0.3,0.1

Type RM Length L Ch R = 1,12096,322,322,322
BEGIN DESCRIPTION:
Mapping XS 26e1dc5c
END DESCRIPTION:
XS GIS Cut Line= 4
      2052878.77     13520180.00      2052790.24     13520237.29
      2052663.50     13520740.76      2052857.94     13520964.70
#Sta/Elev= 30
  4600.7  519.26  4642.2  518.95  4664.7  518.38  4693.6  518.12  4734.7  517.08
  4744.0  517.15  4749.1  516.74  4806.9  515.66  4879.1  513.56  4889.4  513.59
  4899.7  513.94  4930.7  512.76  4954.7  512.44  4982.2  512.55  4987.4  512.32
  4987.9  511.52  4993.3  511.52  4993.8  512.32  5002.8  512.83  5036.9  513.85
  5044.1  514.39  5054.4  514.68  5078.0  514.41  5106.0  514.83  5155.1  516.77
  5160.2  516.74  5224.9  518.73  5406.4  520.25  5442.5  520.84  5521.9  521.50
#Mann=3,-1,0
  4600.7    0.05       0  4987.4    0.03       0  4993.8    0.05       0
Bank Sta=4987.4,4993.8
Exp/Cntr=0.3,0.1

Type RM Length L Ch R = 1,11774,202,202,202
BEGIN DESCRIPTION:
Mapping XS cb24aa03
END DESCRIPTION:
XS GIS Cut Line= 4
      2052988.85     13519947.91      2052760.74     13519956.96
      2052204.97     13520664.79      2052231.67     13520741.34
#Sta/Elev= 30
  4334.6  514.86  4408.5  514.39  4518.6  515.33  4565.4  514.82  4579.9  515.29
  4664.9  515.51  4708.2  516.24  4757.9  516.53  4778.7  515.99  4822.1  515.66
  4871.8  513.99  4942.3  513.05  4956.8  512.28  4979.4  512.68  5000.2  511.44
  5029.1  511.54  5032.2  510.96  5032.7  510.16  5038.1  510.16  5038.6  510.96
  5043.5  511.78  5049.9  511.67  5064.3  512.47  5114.1  514.13  5163.8  514.11
  5234.3  516.20  5292.1  517.18  5370.7  517.90  5426.8  517.27  5543.9  517.35
#Mann=3,-1,0
  4334.6    0.05       0  5032.2    0.03       0  5038.6    0.05       0
Bank Sta=5032.2,5038.6
Exp/Cntr=0.3,0.1

Type RM Length L Ch R = 1,11572,233,233,233
BEGIN DESCRIPTION:
Mapping XS 3a9b6980
END DESCRIPTION:
XS GIS Cut Line= 4
      2053012.35     13519721.62      2052845.83     13519732.48
      2051987.73     13520492.81      2051984.11     13520675.61
#Sta/Elev= 30
  4211.8  517.57  4349.4  516.03  4382.6  516.40  4437.6  512.99  4459.3  512.48
  4586.5  512.80  4657.6  511.75  4678.5  512.76  4686.0  512.08  4692.7  512.94
  4700.2  512.11  4706.9  512.87  4721.1  511.65  4727.8  512.50  4735.3  511.71
  4742.0  512.22  4749.6  511.73  4756.2  512.55  4763.8  512.06  4862.5  512.41
  5001.5  510.86  5002.0  510.06  5007.4  510.06  5007.9  510.86  5068.2  511.02
  5238.0  516.24  5386.9  517.01  5493.1  515.82  5617.4  515.72  5708.0  516.76
#Mann=3,-1,0
  4211.8    0.05       0  5001.5    0.03       0  5007.9    0.05       0
Bank Sta=5001.5,5007.9
Exp/Cntr=0.3,0.1

Type RM Length L Ch R = 1,11339,407,407,407
BEGIN DESCRIPTION:
Mapping XS 6256096b
END DESCRIPTION:
XS GIS Cut Line= 4
      2052786.12     13519687.21      2052507.30     13519784.98
      2051873.68     13520244.80      2051832.23     13520531.36
#Sta/Elev= 30
  4342.2  517.60  4355.0  516.80  4380.7  516.56  4386.0  515.92  4406.4  516.11
  4449.4  514.16  4561.4  515.83  4641.9  515.74  4682.0  514.57  4696.7  514.78
  4732.3  513.41  4747.0  513.53  4767.8  512.57  4832.8  511.67  4875.3  510.10
  4903.9  510.32  4986.5  509.10  4987.0  508.30  4992.4  508.30  4992.9  509.10
  5119.6  510.89  5125.8  511.50  5176.0  512.76  5220.1  513.04  5233.6  513.65
  5261.8  513.37  5362.3  514.42  5423.2  513.42  5521.8  514.91  5710.1  516.51
#Mann=3,-1,0
  4342.2    0.05       0  4986.5    0.03       0  4992.9    0.05       0
Bank Sta=4986.5,4992.9
Exp/Cntr=0.3,0.1

Type RM Length L Ch R = 1,10932,490,490,490
BEGIN DESCRIPTION:
Mapping XS 1cba6d49
END DESCRIPTION:
XS GIS Cut Line= 4
      2052387.51     13519695.63      2052097.53     13519638.33
      2051712.11     13519919.58      2051686.08     13520075.81
#Sta/Elev= 30
  4441.3  518.68  4469.8  518.30  4474.9  518.62  4535.6  517.84  4577.5  516.78
  4596.8  515.90  4623.7  515.73  4628.8  516.12  4647.7  515.93  4708.9  514.40
  4731.3  514.27  4787.0  512.40  4807.8  512.03  4908.3  507.78  4943.8  508.22
  4958.5  507.82  4973.1  507.98  4990.5  506.61  4991.0  505.81  4997.0  505.81
  4997.5  506.61  5000.2  507.45  5029.5  508.92  5058.9  509.31  5086.6  511.18
  5100.6  511.69  5144.6  511.75  5180.1  512.65  5219.5  513.18  5372.4  514.15
#Mann=3,-1,0
  4441.3    0.05       0  4990.5    0.03       0  4997.5    0.05       0
Bank Sta=4990.5,4997.5
Exp/Cntr=0.3,0.1

Type RM Length L Ch R = 1,10442,429,429,429
BEGIN DESCRIPTION:
Mapping XS c05070fb
END DESCRIPTION:
XS GIS Cut Line= 4
      2052227.78     13519419.59      2051913.50     13519306.73
      2051609.68     13519379.65      2051476.00     13519504.65
#Sta/Elev= 30
  4529.6  516.87  4558.5  516.53  4645.4  514.93  4691.9  513.56  4701.6  513.57
  4706.9  513.30  4776.9  511.87  4793.8  511.23  4863.5  509.86  4877.5  509.20
  4903.1  508.48  4919.5  507.35  4924.6  507.31  4944.3  506.18  4975.1  505.59
  4985.4  505.08  4992.2  503.24  4992.7  502.44  4998.7  502.44  4999.2  503.24
  5003.5  503.60  5008.6  503.26  5016.2  505.51  5026.5  506.05  5078.0  506.50
  5149.9  508.21  5246.8  511.47  5296.2  512.01  5346.0  512.09  5359.0  512.34
#Mann=3,-1,0
  4529.6    0.05       0  4992.2    0.03       0  4999.2    0.05       0
Bank Sta=4992.2,4999.2
Exp/Cntr=0.3,0.1

Type RM Length L Ch R = 1,10013,373,373,373
BEGIN DESCRIPTION:
Mapping XS 59d48be4
END DESCRIPTION:
XS GIS Cut Line= 4
      2052361.41     13518848.40      2051859.68     13518772.01
      2051397.88     13519122.70      2051325.25     13519401.10
#Sta/Elev= 30
  4127.5  518.58  4154.2  517.66  4186.5  517.56  4235.1  516.28  4313.6  517.44
  4326.2  518.03  4346.4  517.80  4397.0  517.03  4437.4  515.40  4467.8  515.30
  4488.0  514.49  4528.5  514.54  4647.7  511.85  4812.0  509.85  4891.0  507.38
  4961.7  504.55  4976.3  503.57  4982.6  501.95  4987.2  501.33  4987.7  500.53
  4993.9  500.53  4994.4  501.33  5011.7  504.37  5055.3  503.57  5090.7  504.73
  5118.0  506.26  5168.3  507.27  5218.7  507.55  5372.3  510.82  5502.6  511.85
#Mann=3,-1,0
  4127.5    0.05       0  4987.2    0.03       0  4994.4    0.05       0
Bank Sta=4987.2,4994.4
Exp/Cntr=0.3,0.1

Type RM Length L Ch R = 1,9640,491,491,491
BEGIN DESCRIPTION:
Mapping XS 7a290171
END DESCRIPTION:
XS GIS Cut Line= 4
      2051901.57     13518594.26      2051564.55     13518620.97
      2051074.96     13518983.81      2051037.90     13519190.55
#Sta/Elev= 30
  4277.8  516.35  4294.4  516.35  4364.6  514.10  4384.7  513.99  4414.8  512.71
  4454.9  512.35  4515.1  510.61  4602.0  509.29  4607.0  508.93  4618.7  509.03
  4668.0  507.77  4768.2  506.45  4776.6  506.65  4782.8  506.23  4832.9  505.45
  4889.2  503.14  4926.5  502.98  4976.3  503.59  5000.3  502.67  5000.9  501.87
  5007.1  501.87  5007.6  502.67  5054.1  505.68  5118.8  506.34  5154.2  507.73
  5175.4  508.14  5252.6  509.29  5317.9  509.62  5358.5  510.61  5435.3  510.89
#Mann=3,-1,0
  4277.8    0.05       0  5000.3    0.03       0  5007.6    0.05       0
Bank Sta=5000.3,5007.6
Exp/Cntr=0.3,0.1

Type RM Length L Ch R = 1,9149,555,555,555
BEGIN DESCRIPTION:
Mapping XS 442c7fe8
END DESCRIPTION:
XS GIS Cut Line= 4
      2051578.70     13518301.07      2051363.40     13518294.12
      2050882.50     13518517.65      2050873.48     13518867.81
#Sta/Elev= 30
  4458.6  513.78  4489.5  513.23  4494.5  513.50  4522.3  512.26  4622.4  510.44
  4688.4  508.71  4711.3  507.59  4779.9  505.25  4785.4  505.41  4877.0  502.84
  4968.6  501.66  4991.5  500.58  4993.3  499.48  4993.9  498.68  5000.1  498.68
  5000.6  499.48  5003.1  499.95  5014.1  499.77  5019.9  500.90  5065.6  501.89
  5094.0  502.85  5139.8  504.65  5168.5  506.15  5185.6  506.57  5241.7  506.93
  5271.7  506.56  5391.7  507.60  5511.8  508.09  5531.8  507.86  5554.6  508.21
#Mann=3,-1,0
  4458.6    0.05       0  4993.3    0.03       0  5000.6    0.05       0
Bank Sta=4993.3,5000.6
Exp/Cntr=0.3,0.1

Type RM Length L Ch R = 1,8594,88,88,88
BEGIN DESCRIPTION:
Mapping XS eca009f2
END DESCRIPTION:
XS GIS Cut Line= 4
      2051191.26     13517796.32      2050864.89     13517829.30
      2050654.82     13518221.66      2050673.54     13518311.86
#Sta/Elev= 30
  4473.0  514.68  4507.0  513.26  4519.5  513.41  4539.6  512.23  4650.2  509.70
  4750.7  505.70  4812.3  503.81  4828.5  503.71  4856.1  505.26  4872.4  504.20
  4878.1  504.43  4886.9  503.59  4909.6  500.25  4985.3  497.46  4985.8  496.66
  4992.1  496.66  4992.7  497.46  5020.3  498.74  5034.4  498.44  5064.2  500.08
  5079.7  503.23  5091.8  504.94  5102.4  504.78  5108.0  505.20  5136.4  502.60
  5217.7  504.21  5273.3  504.16  5290.3  504.73  5323.4  504.18  5338.2  504.65
#Mann=3,-1,0
  4473.0    0.05       0  4985.3    0.03       0  4992.7    0.05       0
Bank Sta=4985.3,4992.7
Exp/Cntr=0.3,0.1

Type RM Length L Ch R = 1,8506,51,51,51
BEGIN DESCRIPTION:
Mapping XS 37d57561
END DESCRIPTION:
XS GIS Cut Line= 4
      2051144.38     13517711.25      2050783.30     13517766.80
      2050616.63     13518162.63      2050597.54     13518268.50
#Sta/Elev= 30
  4443.6  514.34  4615.0  509.78  4625.1  509.81  4776.9  504.45  4808.9  504.28
  4820.3  505.87  4828.7  506.12  4861.2  505.60  4867.8  504.58  4873.2  501.98
  4897.0  499.41  4915.3  499.13  4937.2  498.13  4949.9  496.91  4976.9  495.70
  4977.4  494.90  4983.7  494.90  4984.3  495.70  5021.1  497.15  5067.4  499.58
  5074.0  500.31  5089.1  504.15  5097.7  505.18  5110.8  505.63  5121.4  505.86
  5132.5  505.38  5150.6  503.07  5156.0  502.84  5232.7  504.74  5346.0  506.06
#Mann=3,-1,0
  4443.6    0.05       0  4976.9    0.03       0  4984.3    0.05       0
Bank Sta=4976.9,4984.3
Exp/Cntr=0.3,0.1

Type RM Length L Ch R = 1,8455,341,341,341
BEGIN DESCRIPTION:
Mapping XS 20777d50
END DESCRIPTION:
XS GIS Cut Line= 4
      2051094.08     13517600.13      2050746.84     13517728.61
      2050621.84     13518027.22      2050557.87     13518220.86
#Sta/Elev= 30
  4437.2  515.42  4489.3  514.33  4519.7  513.07  4532.2  513.06  4550.1  511.96
  4628.1  509.87  4788.1  503.88  4822.5  503.54  4827.9  502.87  4846.3  503.07
  4851.7  501.81  4857.7  501.91  4875.5  500.81  4880.9  499.77  4904.7  498.54
  4928.5  498.00  4977.8  495.32  4978.3  494.52  4984.6  494.52  4985.2  495.32
  5010.7  496.20  5034.5  497.74  5058.3  498.35  5087.5  499.98  5105.8  501.86
  5127.3  502.60  5167.3  502.89  5294.2  506.06  5307.9  505.85  5335.1  506.30
#Mann=3,-1,0
  4437.2    0.05       0  4977.8    0.03       0  4985.2    0.05       0
Bank Sta=4977.8,4985.2
Exp/Cntr=0.3,0.1

Type RM Length L Ch R = 1,8114,561,561,561
BEGIN DESCRIPTION:
Mapping XS b07d0e2a
END DESCRIPTION:
XS GIS Cut Line= 5
      2050685.38     13517413.11      2050450.98     13517632.32
      2050430.37     13517668.13      2050300.16     13517893.82
      2050278.46     13517964.35
#Sta/Elev= 30
  4640.7  509.80  4706.1  507.91  4769.6  506.52  4797.9  504.48  4826.3  503.52
  4847.3  502.28  4868.8  501.74  4875.6  501.11  4882.9  501.35  4903.9  500.81
  4918.1  500.03  4939.6  499.48  4967.0  497.74  4994.5  496.90  4995.1  496.10
  5001.4  496.10  5002.0  496.90  5041.7  497.68  5047.5  497.42  5122.1  497.84
  5127.9  498.23  5181.0  499.34  5186.8  499.79  5202.6  499.92  5208.4  500.51
  5230.2  501.54  5267.0  502.42  5306.6  503.84  5317.1  503.98  5337.3  503.66
#Mann=3,-1,0
  4640.7    0.05       0  4994.5    0.03       0  5002.0    0.05       0
Bank Sta=4994.5,5002
Exp/Cntr=0.3,0.1

Type RM Length L Ch R = 1,7553,303,303,303
BEGIN DESCRIPTION:
Mapping XS 9ff60ab7
END DESCRIPTION:
XS GIS Cut Line= 4
      2050382.27     13517188.67      2050133.99     13517259.86
      2049906.56     13517462.98      2049929.11     13517780.36
#Sta/Elev= 30
  4552.0  505.92  4601.2  505.31  4674.0  502.67  4726.0  501.74  4834.8  498.88
  4933.4  495.29  4955.2  495.01  4979.5  493.41  4980.1  492.61  4986.4  492.61
  4987.0  493.41  5004.5  494.36  5032.9  494.79  5061.3  496.30  5068.0  497.30
  5089.8  497.45  5110.7  498.89  5113.0  499.50  5163.1  501.68  5168.1  501.27
  5217.5  503.80  5247.6  504.28  5277.6  505.73  5303.8  506.19  5308.8  505.69
  5357.8  506.67  5377.9  506.60  5397.9  507.44  5428.0  507.58  5433.4  507.94
#Mann=3,-1,0
  4552.0    0.05       0  4979.5    0.03       0  4987.0    0.05       0
Bank Sta=4979.5,4987
Exp/Cntr=0.3,0.1

Type RM Length L Ch R = 1,7250,669,669,669
BEGIN DESCRIPTION:
Mapping XS a57992c6
END DESCRIPTION:
XS GIS Cut Line= 4
      2050026.31     13516917.84      2049929.13     13516909.16
      2049602.74     13517511.59      2049708.62     13517676.49
#Sta/Elev= 30
  4521.0  504.10  4592.6  503.91  4618.1  504.64  4683.7  503.41  4699.9  502.43
  4716.1  502.84  4920.9  495.66  4966.4  493.33  4972.8  491.83  4990.9  490.33
  4991.5  489.53  4997.9  489.53  4998.5  490.33  5010.9  492.57  5016.6  492.55
  5023.3  493.77  5038.5  493.44  5068.8  494.53  5120.2  497.27  5193.9  498.15
  5216.6  499.52  5223.9  499.26  5267.6  500.60  5283.8  502.20  5308.7  502.42
  5330.6  503.52  5336.6  503.00  5357.7  503.21  5409.3  504.96  5499.7  506.24
#Mann=3,-1,0
  4521.0    0.05       0  4990.9    0.03       0  4998.5    0.05       0
Bank Sta=4990.9,4998.5
Exp/Cntr=0.3,0.1

Type RM Length L Ch R = 1,6581,786,786,786
BEGIN DESCRIPTION:
Mapping XS bce0f609
END DESCRIPTION:
XS GIS Cut Line= 6
      2049472.51     13516777.22      2049392.67     13516813.68
      2049389.20     13516817.15      2049252.05     13516924.79
      2049168.71     13517421.31      2049250.17     13517509.70
#Sta/Elev= 30
  4584.5  502.02  4647.7  501.43  4802.3  497.66  4842.6  497.46  4847.7  496.63
  4892.3  494.12  4926.0  492.90  4943.0  493.17  4963.3  492.36  4973.4  491.12
  4981.6  483.55  4986.7  485.08  4989.9  483.21  4990.5  482.41  4996.9  482.41
  4997.5  483.21  5003.8  487.10  5024.1  489.08  5034.3  490.92  5042.2  491.63
  5061.2  491.59  5107.9  492.11  5224.1  497.06  5257.3  497.83  5277.6  499.07
  5361.9  500.70  5369.2  501.41  5376.0  500.92  5425.9  502.14  5475.2  502.19
#Mann=5,-1,0
  4584.5    0.05       0  4802.3     0.1       0  4989.9    0.07       0
  4997.5     0.1       0  5061.2    0.05       0
Bank Sta=4989.9,4997.5
Exp/Cntr=0.3,0.1

Type RM Length L Ch R = 1,5795,493,493,493
BEGIN DESCRIPTION:
Mapping XS 2e6236f2
END DESCRIPTION:
XS GIS Cut Line= 4
      2048824.93     13516490.77      2048578.43     13516614.02
      2048474.27     13517138.33      2048576.71     13517324.11
#Sta/Elev= 30
  4384.1  499.36  4402.8  497.69  4425.1  497.09  4497.8  497.05  4609.6  495.94
  4711.7  493.16  4750.8  492.84  4811.0  491.02  4853.1  490.54  4885.0  489.34
  4909.4  487.73  4946.2  487.70  4960.5  487.17  4976.7  485.70  4986.9  483.18
  5006.6  482.97  5007.8  482.42  5008.5  481.62  5014.9  481.62  5015.5  482.42
  5017.5  483.98  5026.9  486.15  5048.1  489.24  5057.7  489.54  5113.9  490.52
  5266.5  494.89  5331.8  495.53  5347.8  496.33  5353.6  495.86  5406.4  496.29
#Mann=5,-1,0
  4384.1    0.05       0  4811.0     0.1       0  5007.8    0.07       0
  5015.5     0.1       0  5026.9    0.05       0
Bank Sta=5007.8,5015.5
Exp/Cntr=0.3,0.1

Type RM Length L Ch R = 1,5302,271,271,271
BEGIN DESCRIPTION:
Mapping XS 3729daf3
END DESCRIPTION:
XS GIS Cut Line= 4
      2048535.03     13516350.13      2048217.32     13516414.37
      2048080.17     13516846.66      2048210.18     13517167.35
#Sta/Elev= 30
  4408.2  495.18  4469.4  494.47  4642.9  493.74  4693.9  492.71  4786.0  492.32
  4827.7  491.65  4869.4  489.28  4911.3  487.83  4951.5  487.06  4974.3  485.64
  4983.8  484.68  4989.0  481.19  4991.4  478.50  4992.0  477.70  4998.5  477.70
  4999.1  478.50  5005.8  481.79  5016.1  483.93  5037.2  486.03  5047.7  485.95
  5068.7  487.13  5085.8  487.45  5198.9  487.79  5235.6  487.77  5241.0  488.18
  5313.3  488.93  5324.3  489.91  5335.1  490.09  5366.9  489.25  5531.9  492.36
#Mann=5,-1,0
  4408.2    0.05       0  4786.0     0.1       0  4991.4    0.07       0
  4999.1     0.1       0  5198.9    0.05       0
Bank Sta=4991.4,4999.1
Exp/Cntr=0.3,0.1

Type RM Length L Ch R = 1,5031,76,76,76
BEGIN DESCRIPTION:
Mapping XS 4b04a73c
END DESCRIPTION:
XS GIS Cut Line= 5
      2048288.33     13516191.89      2048057.87     13516370.27
      2047897.71     13516523.91      2047749.27     13516716.62
      2047725.83     13516875.48
#Sta/Elev= 30
  4559.1  493.10  4734.9  492.97  4778.3  492.22  4784.7  491.00  4791.0  492.35
  4797.2  491.54  4805.5  492.29  4813.7  490.39  4820.0  492.19  4828.1  490.04
  4834.5  491.92  4841.5  489.77  4847.9  489.25  4889.3  487.33  4962.1  483.88
  4976.2  482.77  4986.1  479.78  4991.9  476.98  4992.7  476.18  5001.8  476.18
  5002.7  476.98  5011.5  480.62  5029.8  482.70  5117.9  484.53  5132.5  485.73
  5138.8  484.99  5189.3  486.04  5239.5  487.40  5362.2  490.30  5476.3  490.11
#Mann=11,-1,0
  4559.1    0.05       0  4847.9     0.1       0  4889.3    0.05       0
  4986.1     0.1       0  4991.9    0.07       0  5002.7     0.1       0
  5029.8    0.08       0  5117.9     0.1       0  5189.3    0.08       0
  5239.5     0.1       0  5362.2    0.05       0
Bank Sta=4991.9,5002.7
Exp/Cntr=0.3,0.1

Type RM Length L Ch R = 1,4955,256,256,256
BEGIN DESCRIPTION:
Mapping XS 8f92675f
END DESCRIPTION:
XS GIS Cut Line= 5
      2048274.63     13515968.17      2048000.31     13516315.41
      2047771.14     13516551.52      2047642.67     13516652.22
      2047453.45     13516864.01
#Sta/Elev= 30
  4405.4  492.41  4538.5  491.43  4559.4  492.16  4602.7  491.50  4794.0  492.29
  4858.5  493.54  4907.9  489.35  4917.5  486.85  4922.1  485.79  4946.2  484.42
  4964.5  482.57  4971.7  479.99  4978.7  478.87  4987.4  474.48  4988.3  473.68
  4997.4  473.68  4998.2  474.48  5000.0  475.13  5007.0  474.70  5028.3  482.67
  5035.3  483.44  5092.0  483.97  5127.1  483.60  5185.3  485.56  5230.4  486.79
  5269.6  487.26  5304.8  488.89  5390.0  488.38  5524.6  489.61  5624.2  491.89
#Mann=9,-1,0
  4405.4    0.05       0  4794.0    0.08       0  4917.5    0.05       0
  4946.2    0.08       0  4987.4    0.07       0  4998.2    0.08       0
  5092.0    0.05       0  5185.3    0.08       0  5230.4    0.05       0
Bank Sta=4987.4,4998.2
Exp/Cntr=0.3,0.1

Type RM Length L Ch R = 1,4699,301,301,301
BEGIN DESCRIPTION:
Mapping XS 15bf0bd3
END DESCRIPTION:
XS GIS Cut Line= 4
      2048017.69     13516218.19      2047786.77     13516197.36
      2047505.52     13516544.58      2047446.48     13516794.60
#Sta/Elev= 30
  4591.6  492.17  4634.5  491.38  4686.2  491.91  4704.7  490.93  4765.0  490.73
  4826.6  489.21  4908.9  487.05  4936.3  488.31  4964.9  484.74  4972.8  482.87
  4979.2  482.50  4987.2  475.88  4995.2  475.05  4996.0  474.25  5005.1  474.25
  5006.0  475.05  5008.0  479.72  5014.4  479.65  5036.8  481.91  5064.9  483.07
  5078.4  482.50  5107.1  483.23  5185.5  485.75  5206.5  485.24  5228.6  486.97
  5248.7  487.01  5290.2  486.68  5445.4  488.20  5512.0  489.46  5527.2  490.32
#Mann=5,-1,0
  4591.6    0.05       0  4826.6     0.1       0  4995.2    0.07       0
  5006.0     0.1       0  5248.7    0.05       0
Bank Sta=4995.2,5006
Exp/Cntr=0.3,0.1

Type RM Length L Ch R = 1,4398,1039,1039,1039
BEGIN DESCRIPTION:
Mapping XS 79e41604
END DESCRIPTION:
XS GIS Cut Line= 4
      2048003.80     13516049.78      2047779.82     13516082.77
      2047107.95     13516421.31      2047135.36     13516561.82
#Sta/Elev= 30
  4348.6  491.41  4421.0  491.15  4458.6  489.84  4490.6  489.27  4499.0  489.71
  4569.8  487.81  4711.1  487.62  4737.2  488.24  4811.6  484.55  4817.2  484.88
  4893.9  482.47  4945.5  480.06  4967.8  480.40  4973.4  479.27  4983.5  478.76
  4990.1  477.00  4990.3  474.79  4991.1  473.99  5000.3  473.99  5001.1  474.79
  5003.6  474.98  5005.9  475.16  5012.4  478.69  5018.0  480.66  5028.3  482.06
  5034.7  485.23  5062.6  487.39  5151.9  489.23  5327.3  494.95  5470.5  494.38
#Mann=5,-1,0
  4348.6    0.05       0  4711.1     0.1       0  4990.3    0.07       0
  5001.1     0.1       0  5003.6    0.05       0
Bank Sta=4990.3,5001.1
Exp/Cntr=0.3,0.1

Type RM Length L Ch R = 1,3359,486,486,486
BEGIN DESCRIPTION:
Mapping XS 06e46c85
END DESCRIPTION:
XS GIS Cut Line= 4
      2047913.52     13515497.72      2047722.53     13515318.88
      2047165.24     13515365.76      2047095.80     13515464.72
#Sta/Elev= 30
  4505.8  488.94  4605.7  489.20  4719.0  488.14  4747.4  488.46  4785.4  487.59
  4855.3  484.86  4900.3  484.16  4935.6  482.20  4955.6  478.94  4965.7  477.94
  4985.7  477.50  4990.4  473.09  4991.2  472.29  5000.4  472.29  5001.2  473.09
  5015.1  477.44  5020.1  477.85  5086.1  476.70  5106.2  477.80  5135.0  477.69
  5176.4  479.62  5206.5  481.89  5246.7  482.91  5259.9  483.99  5276.8  483.99
  5306.9  485.50  5316.9  485.28  5324.3  485.84  5333.9  485.58  5447.6  487.86
#Mann=3,-1,0
  4505.8    0.05       0  4990.4    0.03       0  5001.2    0.05       0
Bank Sta=4990.4,5001.2
Exp/Cntr=0.3,0.1

Type RM Length L Ch R = 1,2873,653,653,653
BEGIN DESCRIPTION:
Mapping XS 477a23fc
END DESCRIPTION:
XS GIS Cut Line= 4
      2047922.19     13514987.29      2047701.70     13514851.87
      2047043.71     13514973.40      2046919.33     13515087.41
#Sta/Elev= 30
  4353.9  487.82  4362.2  488.24  4426.0  487.58  4563.3  487.68  4650.0  486.31
  4792.3  482.31  4904.2  482.09  4914.4  481.43  4924.5  480.11  4931.2  478.58
  4955.1  475.78  4989.2  475.34  4990.3  470.84  4991.1  470.04  5000.3  470.04
  5001.1  470.84  5005.9  474.75  5016.1  475.80  5026.2  475.36  5047.2  476.23
  5148.1  481.94  5178.8  482.47  5229.6  484.80  5284.3  485.92  5303.4  487.26
  5345.9  488.12  5352.7  487.79  5360.1  488.61  5402.1  488.96  5450.5  490.45
#Mann=3,-1,0
  4353.9    0.05       0  4990.3    0.03       0  5001.1    0.05       0
Bank Sta=4990.3,5001.1
Exp/Cntr=0.3,0.1

Type RM Length L Ch R = 1,2220,437,437,437
BEGIN DESCRIPTION:
Mapping XS eeb93258
END DESCRIPTION:
XS GIS Cut Line= 4
      2047785.04     13514457.78      2047587.11     13514304.99
      2046852.74     13514325.83      2046661.75     13514454.31
#Sta/Elev= 30
  4393.5  486.47  4509.0  486.71  4545.1  486.55  4552.5  485.80  4558.8  486.48
  4581.5  485.70  4765.7  484.28  4785.7  483.36  4845.7  482.61  4905.8  478.16
  4915.8  476.81  4965.8  472.62  4985.8  470.56  4990.4  469.24  4991.2  468.44
  5000.4  468.44  5001.2  469.24  5005.8  472.04  5025.8  474.12  5035.8  474.22
  5065.8  477.15  5105.8  479.09  5165.9  478.94  5255.9  479.86  5335.9  481.69
  5378.2  483.06  5383.6  483.85  5404.6  483.85  5476.6  486.29  5608.4  488.38
#Mann=3,-1,0
  4393.5    0.05       0  4990.4    0.03       0  5001.2    0.05       0
Bank Sta=4990.4,5001.2
Exp/Cntr=0.3,0.1

Type RM Length L Ch R = 1,1783,300,300,300
BEGIN DESCRIPTION:
Mapping XS 4f2c0f02
END DESCRIPTION:
XS GIS Cut Line= 4
      2047510.76     13513952.58      2047361.42     13513864.02
      2046818.02     13514016.80      2046633.02     13514220.82
#Sta/Elev= 30
  4514.1  484.43  4639.8  485.02  4671.1  483.64  4725.6  483.32  4788.4  481.71
  4817.2  481.87  4829.4  480.57  4850.2  480.04  4895.7  477.08  4902.1  476.00
  4943.7  472.71  4985.2  472.24  4990.2  468.99  4991.0  468.19  5000.2  468.19
  5001.0  468.99  5003.1  470.38  5008.3  472.37  5042.4  472.31  5047.6  473.28
  5068.3  473.92  5130.7  479.22  5194.2  480.94  5260.3  481.39  5317.1  483.30
  5401.6  485.10  5415.8  485.93  5437.4  485.78  5465.7  486.51  5527.6  486.20
#Mann=3,-1,0
  4514.1    0.05       0  4990.2    0.03       0  5001.0    0.05       0
Bank Sta=4990.2,5001
Exp/Cntr=0.3,0.1

Type RM Length L Ch R = 1,1483,248,248,248
BEGIN DESCRIPTION:
Mapping XS e4a6889e
END DESCRIPTION:
XS GIS Cut Line= 4
      2047512.45     13513758.12      2047269.41     13513645.27
      2046668.71     13513740.76      2046547.60     13513920.69
#Sta/Elev= 30
  4399.3  484.04  4421.3  484.53  4518.4  484.67  4581.6  483.10  4650.1  482.87
  4702.3  481.98  4732.5  480.74  4764.5  480.67  4783.1  479.49  4821.7  478.61
  4889.0  474.70  4894.5  473.50  4924.9  471.48  4945.1  470.96  4956.2  471.93
  4975.5  471.68  4985.6  470.65  4990.3  467.43  4991.1  466.63  5000.3  466.63
  5001.1  467.43  5013.4  471.63  5018.5  471.85  5036.2  474.74  5080.7  477.91
  5198.3  478.12  5248.9  479.33  5294.9  479.38  5432.8  482.57  5492.4  482.85
#Mann=3,-1,0
  4399.3    0.05       0  4990.3    0.03       0  5001.1    0.05       0
Bank Sta=4990.3,5001.1
Exp/Cntr=0.3,0.1

Type RM Length L Ch R = 1,1235,369,369,369
BEGIN DESCRIPTION:
Mapping XS 65d342eb
END DESCRIPTION:
XS GIS Cut Line= 4
      2047274.64     13513464.72      2047161.77     13513447.36
      2046689.55     13513468.19      2046606.38     13513610.26
#Sta/Elev= 30
  4644.6  483.92  4684.7  484.12  4694.8  483.26  4725.2  482.86  4745.9  483.28
  4805.6  481.13  4825.6  479.64  4855.7  478.92  4875.7  477.36  4905.7  475.84
  4925.7  473.10  4945.7  471.43  4965.8  470.89  4975.8  471.60  4985.8  470.78
  5000.4  467.76  5001.2  466.96  5010.4  466.96  5011.2  467.76  5015.8  471.10
  5048.3  471.31  5065.9  472.16  5095.9  474.81  5105.9  475.24  5166.0  475.73
  5186.0  475.14  5253.6  477.96  5306.4  479.57  5327.9  479.77  5396.1  478.66
#Mann=3,-1,0
  4644.6    0.05       0  5000.4    0.03       0  5011.2    0.05       0
Bank Sta=5000.4,5011.2
Exp/Cntr=0.3,0.1

Type RM Length L Ch R = 1,866,485,485,485
BEGIN DESCRIPTION:
Mapping XS 2c2ec97c
END DESCRIPTION:
XS GIS Cut Line= 4
      2047137.46     13513094.93      2046979.48     13513030.69
      2046514.20     13513304.99      2046472.58     13513480.15
#Sta/Elev= 30
  4564.7  482.99  4628.8  481.88  4634.2  481.32  4749.9  480.57  4771.4  480.84
  4777.2  481.67  4792.8  482.15  4844.9  480.95  4872.8  479.57  4879.7  478.01
  4903.0  477.17  4937.8  472.97  4974.3  469.95  4984.1  467.47  4989.9  464.98
  5000.2  463.94  5000.9  463.14  5010.2  463.14  5011.0  463.94  5011.4  465.77
  5019.0  468.94  5027.0  470.21  5064.2  470.23  5091.4  471.15  5107.1  470.77
  5144.2  471.54  5216.4  473.94  5272.0  477.02  5297.3  477.60  5455.4  478.19
#Mann=3,-1,0
  4564.7    0.05       0  5000.2    0.03       0  5011.0    0.05       0
Bank Sta=5000.2,5011
Exp/Cntr=0.3,0.1

Type RM Length L Ch R = 1,381,288,288,288
BEGIN DESCRIPTION:
Mapping XS c2a79ab4
END DESCRIPTION:
XS GIS Cut Line= 4
      2046719.09     13512735.55      2046550.66     13512735.55
      2046305.86     13513009.86      2046316.27     13513230.13
#Sta/Elev= 30
  4584.5  476.41  4658.6  475.44  4763.9  475.44  4827.5  473.95  4912.7  473.61
  4954.6  470.11  4968.8  468.37  4976.3  467.96  4983.0  466.45  4990.5  463.00
  4991.8  459.83  4992.5  459.03  5001.8  459.03  5002.6  459.83  5004.7  463.33
  5011.4  467.33  5039.8  468.59  5054.0  468.86  5060.7  468.57  5074.9  469.01
  5096.7  470.72  5110.9  472.54  5120.6  473.12  5125.7  473.93  5145.8  475.51
  5195.8  476.98  5204.5  476.66  5235.9  476.69  5305.9  477.53  5341.1  477.13
#Mann=3,-1,0
  4584.5    0.05       0  4991.8    0.03       0  5002.6    0.05       0
Bank Sta=4991.8,5002.6
Exp/Cntr=0.3,0.1

Type RM Length L Ch R = 1,93,0,0,0
BEGIN DESCRIPTION:
PANTHER Cr 1.0
END DESCRIPTION:
XS GIS Cut Line= 4
      2046913.77     13512400.73      2046332.20     13512639.43
      2046052.25     13512906.36      2046134.72     13513327.39
#Sta/Elev= 30
  4168.7  477.43  4247.1  475.79  4491.7  476.10  4698.0  475.37  4761.9  474.04
  4769.9  474.59  4775.3  473.84  4781.3  474.53  4793.1  474.87  4813.4  473.77
  4848.7  469.62  4969.1  468.39  4976.0  467.78  4983.3  465.75  4990.2  461.54
  4992.0  457.17  4992.8  456.37  5002.1  456.37  5002.8  457.17  5004.4  461.75
  5011.6  465.66  5018.5  466.87  5096.5  469.74  5117.6  471.51  5138.9  471.40
  5193.0  474.21  5227.3  474.22  5273.0  473.49  5407.0  473.86  5613.2  475.83
#Mann=5,-1,0
  4168.7    0.05       0  4781.3     0.1       0  4992.0    0.07       0
  5002.8     0.1       0  5227.3    0.05       0
Bank Sta=4992,5002.8
Exp/Cntr=0.3,0.1

Chan Stop Cuts=-1
