--- Calf Creek.prj (project) ---

Proj Title=Calf Creek Base Level Engineering
Current Plan=p01
Default Exp/Contr=0.3,0.1
English Units
Geom File=g01
Flow File=f01
Plan File=p01
Y Axis Title=Elevation
X Axis Title(PF)=Main Channel Distance
X Axis Title(XS)=Station
BEGIN DESCRIPTION:
Calf Creek
END DESCRIPTION:
DSS Export Rating Curves= 0
DSS Export Rating Curve Sorted= 0
DSS Export Volume Flow Curves= 0
DXF OffsetX= 0
DXF OffsetY= 0
DXF ScaleX= 1
DXF ScaleY= 10

--- Calf Creek.p01 (plan) ---

Plan Title=Multiple Run
Short Identifier=Multiple
Geom File=g01
Flow File=f01
Subcritical Flow
K Sum by GR= 0
Std Step Tol= 0.01
Critical Tol= 0.01
Num of Std Step Trials= 20
Max Error Tol= 0.3
Flow Tol Ratio= 0.001
Split Flow NTrial= 30
Split Flow Tol= 0.02
Split Flow Ratio= 0.02
Log Output Level= 0
Friction Slope Method= 1
Unsteady Friction Slope Method= 2
Unsteady Bridges Friction Slope Method= 1
Parabolic Critical Depth
Global Vel Dist=  1 , 1 , 1
Global Log Level= 0
CheckData=True
Encroach Param= -1, 0, 0, 0
BEGIN DESCRIPTION:
Multiple Run
END DESCRIPTION:

--- Calf Creek.f01 (steady flow) ---

Flow Title=Multiple
Program Version=5.05
Number of Profiles= 7
Profile Names=10-year,25-year,50-year,1pct_min,100-year,1pct_plu,500-year
River Rch & RM=Calf Creek,Reach-1         ,36817
     105     137     163      97     193     385     274
River Rch & RM=Calf Creek,Reach-1         ,36619
     193     262     318     193     385     768     570
River Rch & RM=Calf Creek,Reach-1         ,32659
     287     399     492     302     603    1203     918
River Rch & RM=Calf Creek,Reach-1         ,30376
     362     508     630     389     776    1548    1196
River Rch & RM=Calf Creek,Reach-1         ,19996
     433     613     765     475     947    1889    1475
River Rch & RM=Calf Creek,Reach-1         ,15111
     490     697     873     543    1083    2161    1697
River Rch & RM=Calf Creek,Reach-1         ,3444
     699    1011    1278     802    1601    3194    2554
Boundary for River Rch & Prof#=Calf Creek,Reach-1         , 1
Up Type= 0
Dn Type= 3
Dn Slope=0.00277
Boundary for River Rch & Prof#=Calf Creek,Reach-1         , 2
Up Type= 0
Dn Type= 3
Dn Slope=0.00277
Boundary for River Rch & Prof#=Calf Creek,Reach-1         , 3
Up Type= 0
Dn Type= 3
Dn Slope=0.00277
Boundary for River Rch & Prof#=Calf Creek,Reach-1         , 4
Up Type= 0
Dn Type= 3
Dn Slope=0.00277
Boundary for River Rch & Prof#=Calf Creek,Reach-1         , 5
Up Type= 0
Dn Type= 3
Dn Slope=0.00277
Boundary for River Rch & Prof#=Calf Creek,Reach-1         , 6
Up Type= 0
Dn Type= 3
Dn Slope=0.00277
Boundary for River Rch & Prof#=Calf Creek,Reach-1         , 7
Up Type= 0
Dn Type= 3
Dn Slope=0.00277
DSS Import GetInterval= 0
DSS Import GetPeak= 0
DSS Import FillOption= 0

--- Calf Creek.g01 (geometry) ---

Geom Title=Existing Conditions

River Reach=Calf Creek,Reach-1
Reach XY= 30
      1999073.92     13442929.23      1999740.80     13443164.54
      2000180.80     13443904.54      2001150.80     13443754.54
      2001910.80     13444144.54      2002620.80     13446224.54
      2003320.80     13446294.54      2004180.80     13446994.54
      2004330.80     13447714.54      2004890.80     13447754.54
      2005070.80     13448234.54      2006630.80     13448074.54
      2007280.80     13449134.54      2008610.80     13449634.54
      2008640.80     13450214.54      2009380.06     13449949.39
      2009860.80     13450664.54      2010760.80     13450874.54
      2013192.56     13449394.53      2013416.86     13449617.44
      2013810.80     13448484.54      2014410.80     13447954.54
      2015160.80     13447864.54      2015650.80     13447174.54
      2016238.94     13447747.14      2017690.80     13447624.54
      2017950.80     13447054.54      2018820.80     13446994.54
      2019540.80     13446124.54      2019810.80     13446474.54

Type RM Length L Ch R = 1,36817,198,198,198
BEGIN DESCRIPTION:
Calf Creek 65.0
END DESCRIPTION:
XS GIS Cut Line= 3
      1998565.25     13443541.89      1999175.00     13442975.00
      1999824.97     13442075.04
#Sta/Elev= 30
  4150.0  517.39  4182.4  516.83  4185.3  516.79  4218.1  516.62  4320.6  514.03
  4325.4  513.93  4458.8  511.19  4465.6  511.03  4628.6  509.02  4699.4  508.74
  4890.5  506.01  4907.8  506.48  4968.7  508.01  5004.6  505.37  5031.9  507.66
  5061.1  507.63  5090.5  506.73  5108.4  504.92  5108.9  504.12  5113.9  504.12
  5114.4  504.92  5138.5  505.75  5271.9  507.08  5285.7  507.44  5555.4  509.33
  5626.6  510.69  5698.0  512.96  5863.4  519.65  6028.9  525.16  6092.7  526.35
#Mann=13,-1,0
  4150.0     0.1       0  4182.4    0.08       0  4185.3     0.1       0
  4320.6    0.05       0  4325.4     0.1       0  4458.8    0.05       0
  4465.6     0.1       0  4907.8    0.12       0  5108.4    0.07       0
  5114.4    0.12       0  5138.5     0.1       0  5271.9    0.07       0
  5285.7     0.1       0
Bank Sta=5108.4,5114.4
Exp/Cntr=0.3,0.1

Type RM Length L Ch R = 1,36619,132,132,132
BEGIN DESCRIPTION:
Mapping XS 9bb7508a
END DESCRIPTION:
XS GIS Cut Line= 2
      1998601.73     13443567.91      2000247.51     13442429.93
#Sta/Elev= 30
  4085.4  517.30  4169.0  515.49  4189.8  515.25  4311.9  512.94  4334.9  512.39
  4434.1  511.16  4500.8  510.15  4556.2  509.30  4666.7  508.27  4678.4  508.15
  4832.6  506.50  4922.6  506.32  4998.5  504.94  5022.2  503.64  5022.7  502.84
  5028.5  503.64  5044.8  504.05  5164.3  506.64  5166.9  506.63  5289.1  507.24
  5484.9  507.11  5628.2  509.40  5699.8  512.13  5750.5  511.80  5807.3  513.37
  5822.1  512.51  5858.0  514.00  5872.8  513.04  5893.8  513.97  6086.3  513.83
#Mann=19,-1,0
  4085.4    0.08       0  4169.0     0.1       0  4189.8    0.05       0
  4311.9    0.08       0  4334.9    0.05       0  4434.1    0.08       0
  4500.8     0.1       0  4556.2    0.05       0  4666.7     0.1       0
  4678.4    0.05       0  4832.6     0.1       0  4922.6    0.08       0
  4998.5    0.07       0  5022.2    0.07       0  5028.5    0.07       0
  5044.8    0.05       0  5164.3     0.1       0  5166.9    0.05       0
  5289.1    0.08       0
Bank Sta=5022.2,5028.5
Exp/Cntr=0.3,0.1

Type RM Length L Ch R = 1,36487,471,471,471
BEGIN DESCRIPTION:
Calf Creek 64.0
END DESCRIPTION:
XS GIS Cut Line= 3
      1998683.34     13443678.15      1999503.30     13443081.60
      2000428.12     13442436.83
#Sta/Elev= 30
  4040.0  519.11  4135.7  517.36  4163.1  516.38  4207.9  514.84  4329.2  512.05
  4457.1  509.97  4536.2  509.02  4617.9  508.05  4660.6  507.78  4778.6  505.88
  4785.0  505.85  4938.2  505.25  4985.3  503.22  4985.8  502.42  4991.1  502.42
  4991.6  503.22  5024.0  504.46  5101.2  504.58  5156.5  505.25  5232.2  506.65
  5332.1  506.35  5384.1  506.06  5506.2  507.08  5649.3  509.20  5706.0  510.65
  5777.6  511.35  6051.5  511.96  6072.5  512.64  6108.2  512.67  6181.4  514.71
#Mann=14,-1,0
  4040.0     0.1       0  4135.7    0.08       0  4163.1     0.1       0
  4457.1    0.08       0  4536.2     0.1       0  4617.9    0.08       0
  4660.6     0.1       0  4778.6    0.05       0  4785.0    0.08       0
  4985.3    0.07       0  4991.6    0.08       0  5101.2    0.08       0
  5156.5     0.1       0  5332.1    0.08       0
Bank Sta=4985.3,4991.6
Exp/Cntr=0.3,0.1

Type RM Length L Ch R = 1,36016,466,466,466
BEGIN DESCRIPTION:
Mapping XS 19ec0737
END DESCRIPTION:
XS GIS Cut Line= 2
      1999029.65     13443978.53      2000570.66     13442631.88
#Sta/Elev= 30
  3933.3  519.97  4095.7  516.51  4130.8  515.17  4216.2  513.70  4464.0  507.31
  4591.2  504.85  4747.8  503.68  4825.2  504.13  4946.2  502.88  4960.4  502.32
  4985.7  500.06  4986.2  499.26  4991.5  499.26  4992.0  500.06  4995.5  501.05
  5016.4  502.48  5059.1  504.15  5167.5  504.62  5199.0  504.63  5288.3  505.23
  5484.4  507.62  5506.2  507.26  5576.4  508.02  5612.5  507.41  5633.4  508.76
  5661.9  508.08  5760.6  510.45  5796.6  510.33  5852.8  511.35  5979.8  515.41
#Mann=7,-1,0
  3933.3     0.1       0  4825.2    0.16       0  4985.7    0.07       0
  4992.0    0.16       0  5167.5     0.1       0  5199.0    0.16       0
  5288.3     0.1       0
Bank Sta=4985.7,4992
Exp/Cntr=0.3,0.1

Type RM Length L Ch R = 1,35550,81,81,81
BEGIN DESCRIPTION:
Mapping XS ec7873dd
END DESCRIPTION:
XS GIS Cut Line= 2
      1999345.65     13444100.04      2000727.60     13442773.64
#Sta/Elev= 30
  4298.3  516.79  4421.8  513.39  4442.9  513.88  4457.0  512.15  4485.3  511.03
  4506.4  511.95  4527.8  510.68  4548.8  511.45  4570.2  509.57  4591.3  510.03
  4626.8  508.27  5005.4  500.85  5005.9  500.05  5011.8  500.85  5197.0  503.68
  5297.9  503.00  5355.0  502.08  5438.3  502.72  5492.9  503.05  5578.8  504.61
  5630.8  504.43  5719.2  505.15  5768.8  504.98  5859.7  506.84  5906.7  507.62
  6000.1  509.04  6044.6  510.03  6140.6  512.16  6182.5  513.53  6213.8  515.17
#Mann=18,-1,0
  4298.3    0.05       0  5005.4    0.04       0  5011.8    0.05       0
  5197.0    0.16       0  5297.9    0.05       0  5355.0     0.1       0
  5438.3    0.05       0  5492.9     0.1       0  5578.8    0.05       0
  5630.8     0.1       0  5719.2    0.08       0  5768.8     0.1       0
  5859.7    0.05       0  5906.7     0.1       0  6000.1    0.08       0
  6044.6     0.1       0  6140.6    0.05       0  6182.5     0.1       0
Bank Sta=5005.4,5011.8
Exp/Cntr=0.3,0.1

Type RM Length L Ch R = 1,35469,290,290,290
BEGIN DESCRIPTION:
Mapping XS 7b914c85
END DESCRIPTION:
XS GIS Cut Line= 2
      1999435.94     13444120.85      2000776.24     13442846.53
#Sta/Elev= 30
  4355.5  514.74  4373.1  513.48  4419.1  512.56  4464.9  512.34  4585.4  510.15
  4825.7  503.33  4896.5  502.03  4917.9  502.28  4999.5  500.56  5000.0  499.76
  5005.4  499.76  5005.9  500.56  5087.4  501.30  5158.2  502.73  5207.9  501.62
  5257.3  502.88  5303.8  502.05  5360.7  501.89  5442.3  502.31  5500.5  503.56
  5580.9  503.87  5640.3  504.56  5719.5  505.04  5780.1  505.81  5823.1  505.53
  5919.8  507.21  5999.9  508.39  6135.2  511.91  6199.4  513.69  6204.9  513.75
#Mann=15,-1,0
  4355.5    0.05       0  4419.1     0.1       0  4999.5    0.07       0
  5005.9     0.1       0  5303.8    0.05       0  5360.7     0.1       0
  5442.3    0.05       0  5500.5     0.1       0  5580.9    0.05       0
  5640.3     0.1       0  5719.5    0.08       0  5780.1    0.05       0
  5919.8    0.08       0  6135.2    0.05       0  6199.4    0.08       0
Bank Sta=4999.5,5005.9
Exp/Cntr=0.3,0.1

Type RM Length L Ch R = 1,35179,720,720,720
BEGIN DESCRIPTION:
Mapping XS 0a01de20
END DESCRIPTION:
XS GIS Cut Line= 3
      1999758.87     13444391.65      1999928.99     13444072.25
      2000828.30     13442981.97
#Sta/Elev= 30
  4355.9  513.25  4409.2  513.93  4489.8  511.00  4588.3  509.49  4659.9  507.23
  4798.2  504.62  4869.8  502.02  4890.7  501.87  4897.2  501.18  4933.7  501.29
  4989.7  498.45  5004.1  498.46  5011.9  499.63  5032.7  500.41  5075.8  500.33
  5103.1  500.18  5164.7  497.67  5165.2  496.87  5170.6  496.87  5171.1  497.67
  5189.1  498.69  5230.1  498.62  5240.4  499.20  5267.3  500.76  5331.1  502.21
  5565.6  503.16  5600.8  502.79  5835.3  505.18  5942.2  507.05  6131.1  511.58
#Mann=6,-1,0
  4355.9    0.08       0  4409.2     0.1       0  5164.7    0.07       0
  5171.1     0.1       0  5230.1    0.12       0  5240.4     0.1       0
Bank Sta=5164.7,5171.1
Exp/Cntr=0.3,0.1

Type RM Length L Ch R = 1,34459,429,429,429
BEGIN DESCRIPTION:
Calf Creek 62.0
END DESCRIPTION:
XS GIS Cut Line= 3
      1999748.43     13444641.70      2000422.05     13444214.61
      2000963.73     13443072.22
#Sta/Elev= 30
  3812.9  512.13  3903.5  511.54  3967.1  511.99  4018.8  510.78  4061.1  511.06
  4112.8  509.99  4134.0  510.24  4168.0  509.17  4191.6  509.63  4269.6  507.99
  4329.8  506.42  4343.5  505.49  4519.0  503.72  4656.1  501.39  4787.0  501.66
  4853.5  500.11  4889.0  498.45  4964.2  498.77  4974.5  498.48  4999.5  495.95
  5000.0  495.15  5005.5  495.15  5006.0  495.95  5031.0  498.27  5048.2  498.79
  5167.4  499.55  5190.2  500.38  5417.5  501.16  5650.4  505.37  5874.8  513.66
#Mann=7,-1,0
  3812.9     0.1       0  4168.0    0.05       0  4269.6     0.1       0
  4343.5    0.05       0  4519.0     0.1       0  4999.5    0.07       0
  5006.0     0.1       0
Bank Sta=4999.5,5006
Exp/Cntr=0.3,0.1

Type RM Length L Ch R = 1,34030,547,547,547
BEGIN DESCRIPTION:
Calf Creek 61.0
END DESCRIPTION:
XS GIS Cut Line= 3
      2000646.00     13444953.37      2000852.60     13443985.45
      2001015.79     13443145.18
#Sta/Elev= 30
  3887.1  504.33  3936.6  502.80  4002.6  502.66  4182.0  500.30  4274.0  500.62
  4477.9  499.35  4519.4  499.24  4550.1  497.68  4578.1  497.89  4625.8  497.15
  4642.1  498.23  4670.2  498.74  4703.5  498.10  4764.1  499.20  4818.8  498.95
  4887.5  498.24  4971.1  496.29  5019.5  494.00  5020.0  493.20  5025.5  493.20
  5026.0  494.00  5040.3  495.62  5152.3  498.53  5229.5  499.03  5234.6  498.51
  5274.6  499.76  5441.4  502.22  5519.1  504.55  5661.7  511.27  5732.8  513.43
#Mann=5,-1,0
  3887.1     0.1       0  4477.9    0.05       0  4578.1     0.1       0
  5019.5    0.07       0  5026.0     0.1       0
Bank Sta=5019.5,5026
Exp/Cntr=0.3,0.1

Type RM Length L Ch R = 1,33483,73,73,73
BEGIN DESCRIPTION:
Calf Creek 60.0
END DESCRIPTION:
XS GIS Cut Line= 5
      2000890.79     13445113.95      2001203.30     13444177.29
      2001302.25     13444015.83      2001336.11     13443789.26
      2001457.48     13443608.50
#Sta/Elev= 30
  3700.2  505.87  3720.2  505.24  3727.4  505.84  3732.7  505.17  3741.3  505.82
  3764.3  505.65  3846.7  503.67  3853.8  504.71  3867.8  504.64  4175.2  499.22
  4318.1  497.89  4333.3  498.14  4373.8  496.61  4415.9  496.02  4443.7  496.63
  4500.3  495.71  4649.4  496.49  4756.3  496.06  4857.0  494.52  4903.8  494.51
  4926.4  494.59  4931.4  493.97  4967.8  493.18  4985.8  491.95  4986.3  491.15
  4991.8  491.15  4992.3  491.95  5069.9  496.64  5151.1  500.27  5323.8  506.16
#Mann=7,-1,0
  3700.2     0.1       0  4318.1    0.05       0  4443.7     0.1       0
  4903.8    0.07       0  4967.8     0.1       0  4985.8    0.07       0
  4992.3     0.1       0
Bank Sta=4985.8,4992.3
Exp/Cntr=0.3,0.1

Type RM Length L Ch R = 1,33410,308,308,308
BEGIN DESCRIPTION:
Mapping XS 94e80b3e
END DESCRIPTION:
XS GIS Cut Line= 6
      2000927.24     13445096.58      2001198.09     13444479.37
      2001216.32     13444330.93      2001351.73     13444052.29
      2001388.19     13443859.58      2001520.49     13443771.38
#Sta/Elev= 30
  3756.0  505.67  3815.2  504.44  3833.1  504.79  3838.6  504.33  3856.0  504.98
  3877.9  504.29  3899.7  504.68  3960.9  503.05  4083.1  501.65  4263.1  498.14
  4346.2  497.72  4391.1  496.15  4476.1  495.57  4579.6  495.09  4647.2  495.85
  4708.9  495.48  4714.2  495.96  4838.5  494.40  4945.0  494.21  4970.1  493.76
  4997.4  491.71  4997.9  490.91  5003.4  490.91  5003.9  491.71  5010.8  491.83
  5045.0  494.86  5071.9  495.03  5103.3  497.55  5139.4  498.22  5246.6  502.07
#Mann=7,-1,0
  3756.0     0.1       0  4346.2    0.05       0  4476.1     0.1       0
  4838.5    0.07       0  4945.0     0.1       0  4997.4    0.07       0
  5003.9     0.1       0
Bank Sta=4997.4,5003.9
Exp/Cntr=0.3,0.1

Type RM Length L Ch R = 1,33102,443,443,443
BEGIN DESCRIPTION:
Calf Creek 59.0
END DESCRIPTION:
XS GIS Cut Line= 3
      2000975.00     13445124.99      2001575.00     13444125.00
      2001725.01     13443724.99
#Sta/Elev= 30
  3836.6  506.28  3939.6  504.95  3966.8  503.84  3976.5  504.25  4003.7  503.41
  4019.3  504.00  4128.1  502.66  4209.8  500.60  4375.0  498.32  4463.5  496.31
  4574.0  494.93  4724.8  494.26  4912.7  494.59  4952.2  493.76  4996.6  489.70
  4997.1  488.90  5002.6  488.90  5003.1  489.70  5017.9  490.45  5024.1  492.13
  5042.8  493.50  5128.0  494.35  5244.0  497.85  5274.2  497.98  5329.4  500.36
  5389.9  500.94  5408.6  502.56  5414.9  504.21  5420.2  503.92  5430.0  505.65
#Mann=7,-1,0
  3836.6     0.1       0  4463.5    0.05       0  4574.0     0.1       0
  4912.7    0.07       0  4996.6    0.07       0  5003.1    0.07       0
  5128.0     0.1       0
Bank Sta=4996.6,5003.1
Exp/Cntr=0.3,0.1

Type RM Length L Ch R = 1,32659,419,419,419
BEGIN DESCRIPTION:
Calf Creek 58.0
END DESCRIPTION:
XS GIS Cut Line= 3
      2001127.81     13445023.61      2001975.00     13444225.00
      2002437.65     13443674.70
#Sta/Elev= 30
  3824.2  502.99  3842.5  503.39  3863.5  502.05  3927.5  502.45  4047.6  499.59
  4165.8  497.96  4305.0  495.84  4366.0  494.66  4422.7  492.37  4457.9  493.68
  4528.7  492.27  4578.0  493.17  4606.3  491.96  4634.7  489.65  4670.3  492.43
  4705.5  493.27  4861.6  491.84  4885.3  491.57  4967.2  491.38  4991.7  489.50
  5013.0  486.99  5013.5  486.19  5019.3  486.19  5019.8  486.99  5038.5  490.25
  5045.0  489.89  5131.0  493.18  5244.0  495.81  5563.3  499.67  5707.4  502.57
#Mann=8,-1,0
  3824.2     0.1       0  4165.8    0.05       0  4305.0     0.1       0
  4861.6    0.12       0  4885.3    0.07       0  5013.0    0.07       0
  5019.8    0.07       0  5131.0     0.1       0
Bank Sta=5013,5019.8
Exp/Cntr=0.3,0.1

Type RM Length L Ch R = 1,32240,540,540,540
BEGIN DESCRIPTION:
Calf Creek 57.0
END DESCRIPTION:
XS GIS Cut Line= 3
      2001250.19     13445057.48      2002049.65     13444596.56
      2002896.04     13444276.23
#Sta/Elev= 30
  4011.8  502.44  4121.2  500.55  4127.0  499.68  4148.5  499.29  4224.5  498.82
  4348.4  496.71  4662.7  491.50  4698.4  490.05  4727.4  487.39  4743.2  487.62
  4786.3  490.44  4829.4  490.69  4934.6  488.73  4961.7  487.26  4984.9  487.80
  4993.8  487.41  5000.9  485.75  5001.4  484.95  5007.3  484.95  5007.8  485.75
  5025.9  486.74  5047.3  489.39  5079.3  488.70  5107.9  489.69  5170.2  492.22
  5405.3  494.68  5575.6  497.31  5605.8  498.84  5817.1  503.78  5839.6  504.89
#Mann=7,-1,0
  4011.8     0.1       0  4224.5    0.05       0  4348.4     0.1       0
  5000.9    0.07       0  5007.8     0.1       0  5107.9    0.16       0
  5170.2     0.1       0
Bank Sta=5000.9,5007.8
Exp/Cntr=0.3,0.1

Type RM Length L Ch R = 1,31700,250,250,250
BEGIN DESCRIPTION:
Calf Creek 56.0
END DESCRIPTION:
XS GIS Cut Line= 3
      2001372.57     13445231.97      2002175.00     13445075.00
      2002974.98     13444625.01
#Sta/Elev= 30
  4183.3  502.79  4297.6  501.17  4398.4  498.36  4399.7  498.33  4420.1  498.82
  4609.5  494.38  4848.1  490.73  4946.1  487.70  4960.2  486.26  4970.1  484.09
  4975.2  485.28  4986.9  482.08  4987.5  481.28  4994.0  481.28  4994.7  482.08
  5008.9  483.53  5014.6  482.91  5030.6  486.14  5036.3  485.18  5046.5  485.58
  5052.3  484.41  5095.6  486.38  5127.2  486.12  5161.6  488.10  5203.1  488.99
  5316.8  490.68  5413.7  490.74  5624.7  494.36  5829.9  501.47  5918.8  503.68
#Mann=8,-1,0
  4183.3     0.1       0  4297.6    0.08       0  4398.4    0.05       0
  4399.7     0.1       0  4946.1    0.16       0  4986.9    0.07       0
  4994.7    0.16       0  5203.1     0.1       0
Bank Sta=4986.9,4994.7
Exp/Cntr=0.3,0.1

Type RM Length L Ch R = 1,31450,362,362,362
BEGIN DESCRIPTION:
Calf Creek 55.0
END DESCRIPTION:
XS GIS Cut Line= 3
      2001492.36     13445617.39      2002239.75     13445307.49
      2003229.37     13444841.34
#Sta/Elev= 30
  4149.0  501.58  4227.6  500.07  4274.5  500.33  4342.3  498.76  4368.4  497.64
  4380.9  498.58  4399.3  498.53  4428.6  496.90  4450.1  496.81  4457.9  497.71
  4476.4  496.84  4552.4  496.06  4595.7  494.58  4718.4  492.31  4742.3  491.20
  4896.8  488.55  4978.1  486.57  4986.0  485.51  4995.3  482.66  4997.0  481.13
  4997.6  480.33  5004.1  480.33  5004.8  481.13  5046.4  485.33  5092.0  485.24
  5151.8  487.39  5228.3  488.25  5273.4  487.80  5536.0  490.95  6052.0  502.96
#Mann=7,-1,0
  4149.0     0.1       0  4342.3    0.05       0  4450.1     0.1       0
  4896.8    0.16       0  4997.0    0.07       0  5004.8    0.16       0
  5228.3     0.1       0
Bank Sta=4997,5004.8
Exp/Cntr=0.3,0.1

Type RM Length L Ch R = 1,31088,48,48,48
BEGIN DESCRIPTION:
Mapping XS f3f2af8c
END DESCRIPTION:
XS GIS Cut Line= 6
      2001757.98     13445708.54      2002198.09     13445580.93
      2002382.98     13445565.31      2002445.48     13445570.51
      2002599.13     13445494.99      2003336.12     13445091.34
#Sta/Elev= 30
  4293.3  496.49  4299.7  497.09  4818.7  487.74  4848.8  491.17  4912.2  479.86
  4945.2  477.84  4945.9  477.04  4953.0  477.84  4988.9  480.14  4997.0  483.23
  5002.9  481.04  5019.8  482.86  5025.4  480.19  5042.3  481.99  5047.9  479.55
  5064.8  481.13  5070.3  478.92  5087.2  480.97  5092.8  478.80  5109.7  480.75
  5121.4  479.68  5123.4  479.87  5154.7  481.12  5160.2  479.23  5226.0  490.75
  5236.2  488.50  5242.1  486.50  5263.9  486.08  5360.1  486.77  6011.3  500.60
#Mann=8,-1,0
  4293.3    0.05       0  4299.7     0.1       0  4912.2    0.12       0
  4945.2    0.07       0  4953.0    0.12       0  5121.4     0.1       0
  5123.4    0.07       0  5236.2     0.1       0
Bank Sta=4945.2,4953
Exp/Cntr=0.3,0.1

Type RM Length L Ch R = 1,31040,36,36,36
BEGIN DESCRIPTION:
Mapping XS 27770e25
END DESCRIPTION:
XS GIS Cut Line= 5
      2001698.10     13445773.64      2002195.48     13445625.20
      2002409.03     13445614.79      2002557.46     13445606.97
      2003398.64     13445114.77
#Sta/Elev= 30
  4207.4  498.54  4274.7  496.05  4291.5  496.83  4548.5  492.95  4572.2  493.46
  4776.0  488.09  4796.1  488.37  4846.1  491.77  4986.1  492.32  5006.3  492.20
  5026.3  490.02  5031.3  492.08  5046.4  491.59  5085.0  488.49  5097.3  488.20
  5103.1  490.92  5118.8  488.93  5124.6  490.28  5140.2  487.89  5161.7  486.47
  5198.9  485.66  5216.5  484.33  5217.1  483.53  5223.6  483.53  5224.3  484.33
  5263.4  485.92  5322.0  485.71  5491.6  488.40  5593.9  491.50  6063.5  501.16
#Mann=6,-1,0
  4207.4    0.05       0  4274.7     0.1       0  4986.1    0.12       0
  5085.0     0.1       0  5216.5    0.07       0  5224.3     0.1       0
Bank Sta=5216.5,5224.3
Exp/Cntr=0.3,0.1

Type RM Length L Ch R = 1,31004,188,188,188
BEGIN DESCRIPTION:
Mapping XS 33a3773c
END DESCRIPTION:
XS GIS Cut Line= 6
      2001729.32     13445817.92      2002239.75     13445661.66
      2002450.69     13445646.04      2002523.61     13445640.83
      2002640.80     13445596.56      2003375.13     13445151.27
#Sta/Elev= 30
  4218.8  498.08  4251.9  496.63  4315.1  495.91  4601.2  492.27  4695.4  489.29
  4757.9  489.05  4788.0  487.11  4858.1  486.22  4898.3  484.41  4906.9  484.89
  4911.9  487.44  4918.3  487.39  5014.7  481.58  5015.3  480.78  5022.5  481.58
  5060.1  482.80  5072.4  484.90  5090.7  486.07  5127.0  486.60  5253.7  485.04
  5443.7  486.90  5480.5  487.56  5486.4  488.55  5517.4  488.23  5523.2  489.24
  5538.7  488.97  5544.5  490.24  5560.0  489.79  5588.4  491.25  6021.3  500.19
#Mann=7,-1,0
  4218.8     0.1       0  4251.9    0.05       0  4315.1     0.1       0
  5014.7    0.07       0  5022.5     0.1       0  5072.4    0.07       0
  5090.7     0.1       0
Bank Sta=5014.7,5022.5
Exp/Cntr=0.3,0.1

Type RM Length L Ch R = 1,30816,440,440,440
BEGIN DESCRIPTION:
Calf Creek 54.0
END DESCRIPTION:
XS GIS Cut Line= 3
      2001724.96     13445925.00      2002525.00     13445825.00
      2003484.08     13445229.66
#Sta/Elev= 30
  4184.1  498.33  4216.8  497.65  4264.8  495.41  4295.0  496.08  4316.3  495.37
  4607.4  489.36  4705.7  488.50  4748.5  486.73  4829.1  485.26  4952.6  483.88
  4970.2  483.19  4980.3  481.46  4987.8  479.17  5000.0  478.21  5000.7  477.41
  5007.2  477.41  5007.8  478.21  5025.7  479.54  5034.7  482.24  5049.2  484.59
  5077.2  486.24  5092.5  485.09  5119.8  484.69  5187.0  485.13  5244.9  484.08
  5260.2  485.17  5296.4  484.05  5354.7  484.39  5470.5  486.06  6119.2  500.53
#Mann=5,-1,0
  4184.1     0.1       0  4216.8    0.08       0  4316.3     0.1       0
  5000.0    0.07       0  5007.8     0.1       0
Bank Sta=5000,5007.8
Exp/Cntr=0.3,0.1

Type RM Length L Ch R = 1,30376,510,510,510
BEGIN DESCRIPTION:
Calf Creek 53.0
END DESCRIPTION:
XS GIS Cut Line= 3
      2001804.83     13446419.48      2002539.23     13446312.70
      2003324.99     13445575.01
#Sta/Elev= 30
  4137.8  494.42  4242.8  492.23  4339.8  490.89  4643.2  487.79  4689.4  485.57
  4734.2  486.36  4744.3  486.10  4759.6  483.55  4829.7  481.66  4845.3  483.84
  4875.3  481.66  4953.2  481.41  4960.1  480.48  4981.6  482.89  4995.7  477.62
  5005.7  477.32  5006.4  476.52  5014.0  477.32  5045.1  480.38  5066.1  480.28
  5087.6  482.46  5243.4  483.76  5349.4  481.76  5363.5  479.94  5377.7  481.26
  5391.9  480.43  5441.2  481.69  5526.2  487.38  5597.0  489.96  5957.7  494.34
#Mann=5,-1,0
  4137.8     0.1       0  4242.8    0.05       0  4339.8     0.1       0
  5005.7    0.07       0  5014.0     0.1       0
Bank Sta=5005.7,5014
Exp/Cntr=0.3,0.1

Type RM Length L Ch R = 1,29866,497,497,497
BEGIN DESCRIPTION:
Calf Creek 52.0
END DESCRIPTION:
XS GIS Cut Line= 3
      2002307.45     13447057.51      2003002.78     13446297.08
      2003262.74     13445829.15
#Sta/Elev= 30
  3979.7  495.93  4070.3  493.97  4112.3  493.23  4251.9  489.99  4298.1  489.38
  4432.5  485.01  4878.4  483.32  4949.3  481.05  4970.9  477.15  4977.7  477.62
  4991.9  476.36  5004.0  474.15  5004.7  473.35  5011.6  473.35  5012.3  474.15
  5014.2  474.15  5021.6  478.46  5035.4  480.69  5092.6  481.65  5152.0  480.30
  5241.3  481.17  5271.0  479.78  5287.0  476.70  5292.7  474.38  5298.5  474.27
  5314.4  480.69  5330.5  482.88  5357.9  488.53  5379.7  491.40  5545.4  494.34
#Mann=6,-1,0
  3979.7    0.05       0  4070.3     0.1       0  4112.3    0.05       0
  4251.9     0.1       0  5004.0    0.07       0  5012.3     0.1       0
Bank Sta=5004,5012.3
Exp/Cntr=0.3,0.1

Type RM Length L Ch R = 1,29369,581,581,581
BEGIN DESCRIPTION:
Calf Creek 51.0
END DESCRIPTION:
XS GIS Cut Line= 3
      2002617.34     13447338.77      2003257.98     13446518.43
      2003687.12     13446159.52
#Sta/Elev= 30
  3791.1  494.78  3872.8  492.98  4004.6  489.51  4090.4  487.20  4090.5  487.20
  4219.4  483.84  4233.9  484.09  4404.9  481.64  4468.4  481.43  4640.0  483.13
  4675.2  482.57  4753.9  482.76  4860.7  478.52  4910.1  479.23  4938.8  478.74
  4967.4  476.52  4988.2  476.06  4996.0  474.06  4998.3  471.89  4999.0  471.09
  5006.0  471.09  5006.8  471.89  5010.3  472.48  5016.8  474.92  5023.6  478.73
  5031.1  479.15  5037.7  480.40  5059.8  481.72  5130.0  485.04  5391.4  493.91
#Mann=7,-1,0
  3791.1     0.1       0  3872.8    0.05       0  4004.6     0.1       0
  4090.4    0.05       0  4090.5     0.1       0  4998.3    0.07       0
  5006.8     0.1       0
Bank Sta=4998.3,5006.8
Exp/Cntr=0.3,0.1

Type RM Length L Ch R = 1,28788,503,503,503
BEGIN DESCRIPTION:
Calf Creek 50.0
END DESCRIPTION:
XS GIS Cut Line= 3
      2002875.03     13447524.97      2003675.00     13446875.00
      2003775.00     13446224.98
#Sta/Elev= 30
  3928.7  495.86  4014.1  493.88  4028.5  492.94  4106.8  490.67  4162.8  489.74
  4313.0  484.47  4461.6  480.68  4639.1  478.59  4830.8  479.88  4895.0  479.67
  4923.5  478.30  4945.8  476.20  4952.2  476.57  4956.2  474.26  4962.0  474.26
  4969.6  475.36  4988.5  471.93  4989.3  469.79  4990.1  468.99  4997.1  468.99
  4997.8  469.79  5010.0  473.93  5030.3  476.72  5050.5  476.80  5070.7  477.87
  5293.3  481.09  5383.1  485.61  5388.2  485.09  5607.0  494.67  5617.1  494.54
#Mann=3,-1,0
  3928.7     0.1       0  4989.3    0.07       0  4997.8     0.1       0
Bank Sta=4989.3,4997.8
Exp/Cntr=0.3,0.1

Type RM Length L Ch R = 1,28285,272,272,272
BEGIN DESCRIPTION:
Calf Creek 49.0
END DESCRIPTION:
XS GIS Cut Line= 3
      2002925.03     13447574.98      2004125.00     13446975.00
      2004424.63     13446544.51
#Sta/Elev= 30
  3653.9  495.94  3818.8  490.76  3869.1  490.31  3908.2  488.13  4078.7  483.24
  4338.7  478.12  4458.8  477.17  4570.6  478.24  4808.2  477.63  4936.8  475.99
  4981.5  471.78  4987.1  470.55  4988.5  468.79  4989.2  467.99  4996.2  467.99
  4997.0  468.79  5002.9  469.32  5009.0  471.76  5032.1  473.35  5038.7  475.12
  5044.8  473.12  5053.5  475.70  5059.6  474.04  5068.4  474.42  5074.5  474.98
  5080.8  477.05  5104.2  478.92  5318.9  486.46  5361.0  488.75  5520.0  493.60
#Mann=3,-1,0
  3653.9     0.1       0  4988.5    0.07       0  4997.0     0.1       0
Bank Sta=4988.5,4997
Exp/Cntr=0.3,0.1

Type RM Length L Ch R = 1,28013,837,837,837
BEGIN DESCRIPTION:
Calf Creek 48.0
END DESCRIPTION:
XS GIS Cut Line= 3
      2003273.60     13448153.86      2003901.21     13447398.64
      2004720.73     13446847.09
#Sta/Elev= 30
  3608.7  490.29  3622.7  489.38  3879.2  486.31  4169.6  480.10  4297.2  479.25
  4319.3  477.58  4354.5  478.74  4582.3  476.16  4588.8  474.86  4603.7  474.50
  4631.4  476.61  4747.7  475.53  4855.6  476.33  4891.6  475.12  4956.8  475.01
  4969.6  474.75  4978.6  471.95  4984.6  471.75  4993.0  469.06  5001.4  468.28
  5002.1  467.48  5009.1  467.48  5009.9  468.28  5014.6  470.37  5020.6  470.72
  5035.6  474.79  5077.6  477.90  5158.5  479.08  5353.5  484.16  5578.5  491.20
#Mann=3,-1,0
  3608.7     0.1       0  5001.4    0.07       0  5009.9     0.1       0
Bank Sta=5001.4,5009.9
Exp/Cntr=0.3,0.1

Type RM Length L Ch R = 1,27176,629,629,629
BEGIN DESCRIPTION:
Calf Creek 47.0
END DESCRIPTION:
XS GIS Cut Line= 3
      2003925.00     13448375.00      2004450.69     13447875.20
      2004898.59     13446963.78
#Sta/Elev= 30
  4117.9  485.56  4139.1  483.92  4372.5  478.09  4683.6  474.87  4842.8  472.02
  4876.1  472.41  4921.5  472.38  4957.8  471.46  4974.7  469.28  4988.3  468.58
  4992.7  465.14  4993.6  464.34  5000.8  464.34  5001.6  465.14  5019.6  472.18
  5032.9  472.76  5092.6  472.34  5109.6  473.16  5177.0  473.88  5222.0  473.11
  5227.5  473.69  5233.5  473.05  5311.5  473.59  5323.0  474.31  5378.3  474.52
  5502.8  477.05  5750.1  485.36  5772.6  486.87  5795.1  487.03  5858.8  489.75
#Mann=5,-1,0
  4117.9     0.1       0  4876.1    0.07       0  4992.7    0.07       0
  5001.6    0.07       0  5092.6     0.1       0
Bank Sta=4992.7,5001.6
Exp/Cntr=0.3,0.1

Type RM Length L Ch R = 1,26547,398,398,398
BEGIN DESCRIPTION:
Calf Creek 46.0
END DESCRIPTION:
XS GIS Cut Line= 3
      2004187.64     13448599.19      2005054.86     13447802.29
      2005225.00     13447125.00
#Sta/Elev= 30
  4004.3  484.77  4090.4  481.57  4097.2  479.66  4106.8  478.73  4111.4  477.20
  4118.7  477.05  4147.1  476.99  4153.9  478.61  4210.6  478.37  4247.7  476.48
  4415.9  474.39  4692.1  473.79  4812.4  469.30  4847.5  470.45  4875.9  469.62
  4904.2  466.31  4925.2  469.60  4967.8  469.93  4996.1  467.31  5005.8  463.87
  5006.7  463.07  5014.7  463.87  5031.9  470.47  5052.8  471.88  5245.2  470.26
  5375.2  471.94  5574.4  477.41  5663.9  481.71  5780.1  484.94  5880.4  489.95
#Mann=5,-1,0
  4004.3     0.1       0  4106.8    0.05       0  4247.7     0.1       0
  5005.8    0.07       0  5014.7     0.1       0
Bank Sta=5005.8,5014.7
Exp/Cntr=0.3,0.1

Type RM Length L Ch R = 1,26149,318,318,318
BEGIN DESCRIPTION:
Calf Creek 45.0
END DESCRIPTION:
XS GIS Cut Line= 3
      2004324.98     13448775.01      2005125.00     13448225.00
      2005424.98     13447425.04
#Sta/Elev= 30
  4067.8  483.39  4197.7  478.27  4341.1  474.37  4478.3  474.69  4551.8  473.66
  4571.2  474.48  4629.0  472.77  4771.7  472.81  4795.1  472.45  4816.1  470.48
  4822.1  472.41  4880.9  472.17  4953.4  470.48  4959.5  468.70  4974.4  470.42
  4989.3  466.39  4990.9  464.74  4991.7  463.94  4999.8  464.74  5048.4  468.27
  5084.0  467.53  5102.7  469.70  5164.1  468.54  5209.5  469.79  5335.0  468.93
  5497.9  472.28  5583.3  472.24  5596.7  473.58  5797.8  478.25  5893.0  482.21
#Mann=6,-1,0
  4067.8     0.1       0  4478.3    0.05       0  4551.8    0.08       0
  4629.0     0.1       0  4990.9    0.07       0  4999.8     0.1       0
Bank Sta=4990.9,4999.8
Exp/Cntr=0.3,0.1

Type RM Length L Ch R = 1,25831,575,575,575
BEGIN DESCRIPTION:
Calf Creek 44.0
END DESCRIPTION:
XS GIS Cut Line= 3
      2004475.01     13449374.98      2005333.50     13448325.72
      2005567.87     13447474.20
#Sta/Elev= 30
  3591.2  483.55  3619.2  483.53  3818.7  477.40  3853.9  477.62  3875.4  476.21
  3882.6  477.11  3889.1  476.23  3917.8  475.73  4159.7  472.40  4323.3  470.96
  4728.2  471.07  4778.4  472.04  4809.8  471.00  4862.2  471.47  4949.9  469.33
  4972.5  466.40  4999.5  464.88  5006.9  465.44  5007.6  464.03  5008.4  463.23
  5015.7  463.23  5016.6  464.03  5020.3  466.53  5030.6  467.12  5046.5  469.63
  5072.1  467.93  5165.5  467.68  5455.9  471.08  5727.9  477.41  5830.1  481.06
#Mann=5,-1,0
  3591.2     0.1       0  4809.8    0.05       0  4862.2     0.1       0
  5007.6    0.07       0  5016.6     0.1       0
Bank Sta=5007.6,5016.6
Exp/Cntr=0.3,0.1

Type RM Length L Ch R = 1,25256,639,639,639
BEGIN DESCRIPTION:
Calf Creek 43.0
END DESCRIPTION:
XS GIS Cut Line= 3
      2004935.09     13449549.64      2005625.17     13448466.35
      2005825.00     13447475.01
#Sta/Elev= 30
  3514.0  478.70  3691.0  473.52  3806.2  471.41  4030.5  469.56  4306.4  469.16
  4574.7  470.39  4790.7  469.56  4840.6  467.57  4887.7  467.91  4963.0  467.25
  4971.4  464.24  4999.3  461.31  5000.1  460.51  5007.5  460.51  5008.4  461.31
  5014.0  464.77  5022.2  465.51  5027.3  467.43  5054.8  465.00  5065.0  466.36
  5085.4  466.81  5116.0  466.57  5128.9  465.19  5290.9  468.76  5433.8  469.30
  5530.3  474.17  5758.7  480.59  5784.3  483.31  5789.4  482.59  5809.7  483.21
#Mann=6,-1,0
  3514.0     0.1       0  4790.7    0.05       0  4887.7     0.1       0
  4999.3    0.07       0  5008.4     0.1       0  5290.9    0.05       0
Bank Sta=4999.3,5008.4
Exp/Cntr=0.3,0.1

Type RM Length L Ch R = 1,24617,846,846,846
BEGIN DESCRIPTION:
Mapping XS 3611166e
END DESCRIPTION:
XS GIS Cut Line= 3
      2005099.56     13449495.86      2006012.76     13448509.75
      2006474.46     13447589.82
#Sta/Elev= 30
  3213.8  473.76  3437.5  469.47  3657.0  468.32  4456.4  468.64  4498.9  467.95
  4513.1  468.62  4628.4  467.48  4646.7  466.87  4666.3  465.33  4688.6  465.29
  4697.4  467.13  4912.0  465.46  4973.4  463.31  4979.0  463.85  4988.3  462.65
  4996.8  459.43  4997.6  458.63  5005.0  458.63  5005.9  459.43  5018.0  462.14
  5055.4  464.49  5090.6  464.37  5202.3  466.93  5291.7  470.78  5301.6  472.43
  5324.0  472.18  5336.3  473.47  5350.6  473.65  5509.4  480.70  5587.1  482.36
#Mann=6,-1,0
  3213.8     0.1       0  4628.4    0.05       0  4646.7     0.1       0
  4996.8    0.07       0  5005.9     0.1       0  5350.6    0.05       0
Bank Sta=4996.8,5005.9
Exp/Cntr=0.3,0.1

Type RM Length L Ch R = 1,23771,115,115,115
BEGIN DESCRIPTION:
Mapping XS e4cfa2fb
END DESCRIPTION:
XS GIS Cut Line= 5
      2005054.44     13449596.54      2006495.40     13448318.78
      2006769.70     13448343.08      2006870.40     13448315.31
      2007247.65     13448059.19
#Sta/Elev= 30
  2756.1  476.51  2885.2  472.57  2977.2  471.30  2991.4  470.23  3182.9  468.50
  4373.0  467.31  4514.4  465.61  4577.9  463.31  4655.7  464.64  4932.6  461.22
  4962.9  461.67  4994.0  459.79  5003.5  456.44  5004.4  455.64  5011.8  455.64
  5012.6  456.44  5025.1  459.12  5035.5  459.59  5042.4  461.66  5047.6  459.71
  5061.6  462.23  5072.4  460.80  5102.2  461.81  5123.2  463.28  5144.2  466.41
  5159.2  465.39  5174.1  466.73  5180.2  468.23  5217.4  469.73  5517.8  480.77
#Mann=4,-1,0
  2756.1     0.1       0  5003.5    0.07       0  5012.6     0.1       0
  5217.4    0.05       0
Bank Sta=5003.5,5012.6
Exp/Cntr=0.3,0.1

Type RM Length L Ch R = 1,23656,483,483,483
BEGIN DESCRIPTION:
Calf Creek 42.0
END DESCRIPTION:
XS GIS Cut Line= 5
      2005096.95     13449642.57      2006443.31     13448444.65
      2006630.81     13448439.44      2006794.88     13448462.88
      2007290.51     13448125.52
#Sta/Elev= 30
  2801.1  476.24  2876.2  473.64  3039.2  469.73  3088.5  469.78  3180.5  468.53
  3719.0  467.34  4356.2  467.69  4683.5  464.23  4765.0  462.15  4785.0  462.43
  4790.4  463.31  4816.9  462.91  4962.2  460.88  4992.1  459.86  4998.1  459.52
  5000.5  456.09  5001.4  455.29  5008.8  455.29  5009.6  456.09  5028.0  461.12
  5034.0  459.51  5049.0  460.26  5063.9  460.08  5099.8  461.98  5120.8  463.99
  5186.5  465.36  5243.5  468.80  5292.8  470.41  5380.1  473.58  5556.1  477.99
#Mann=6,-1,0
  2801.1     0.1       0  4683.5    0.05       0  4816.9     0.1       0
  5000.5    0.07       0  5009.6     0.1       0  5292.8    0.05       0
Bank Sta=5000.5,5009.6
Exp/Cntr=0.3,0.1

Type RM Length L Ch R = 1,23173,510,510,510
BEGIN DESCRIPTION:
Calf Creek 41.0
END DESCRIPTION:
XS GIS Cut Line= 3
      2005714.16     13450221.54      2007025.00     13448825.00
      2007345.65     13448181.64
#Sta/Elev= 30
  3120.0  474.85  3245.5  472.05  3471.8  465.18  3627.4  463.33  3669.9  464.39
  3677.2  464.25  3684.1  462.88  3726.6  464.55  3995.2  463.16  4448.0  465.39
  4469.5  464.63  4759.6  464.00  4851.5  463.08  4918.6  461.28  4943.3  459.58
  4958.8  459.61  4985.8  460.21  4993.1  459.72  5002.7  456.97  5003.6  456.17
  5011.0  456.17  5011.9  456.97  5031.9  459.15  5047.4  459.51  5133.3  459.89
  5273.2  462.18  5497.0  468.84  5513.8  468.26  5584.4  471.82  5754.2  477.02
#Mann=7,-1,0
  3120.0     0.1       0  4918.6    0.05       0  4958.8    0.12       0
  5002.7    0.07       0  5011.9    0.12       0  5047.4     0.1       0
  5584.4    0.05       0
Bank Sta=5002.7,5011.9
Exp/Cntr=0.3,0.1

Type RM Length L Ch R = 1,22663,429,429,429
BEGIN DESCRIPTION:
Calf Creek 40.0
END DESCRIPTION:
XS GIS Cut Line= 3
      2006075.01     13450324.99      2007275.00     13449125.00
      2007703.24     13448389.07
#Sta/Elev= 30
  3305.6  471.31  3489.4  466.00  3758.1  460.89  3786.4  461.78  3814.7  460.16
  3913.7  462.11  4055.1  461.09  4380.4  463.27  4733.9  462.54  4877.3  460.43
  4974.4  458.41  4980.5  456.92  4994.5  454.83  4995.4  454.03  5003.7  454.83
  5010.8  454.99  5016.3  457.04  5047.7  458.81  5222.5  459.78  5251.3  458.43
  5267.0  460.36  5272.8  459.52  5288.5  460.67  5427.5  461.49  5454.8  460.58
  5477.0  462.12  5492.1  461.58  5507.8  463.31  5653.1  465.65  5854.1  468.66
#Mann=7,-1,0
  3305.6     0.1       0  4877.3    0.05       0  4980.5    0.12       0
  4994.5    0.07       0  5003.7    0.12       0  5010.8     0.1       0
  5653.1    0.05       0
Bank Sta=4994.5,5003.7
Exp/Cntr=0.3,0.1

Type RM Length L Ch R = 1,22234,401,401,401
BEGIN DESCRIPTION:
Calf Creek 39.0
END DESCRIPTION:
XS GIS Cut Line= 3
      2006724.99     13450475.02      2007625.00     13449275.00
      2008082.19     13448416.02
#Sta/Elev= 30
  3524.4  475.31  3581.7  470.51  3681.7  464.50  3781.7  460.88  3924.4  457.89
  3974.4  458.92  3981.7  457.28  3996.3  458.36  4146.3  460.65  4252.5  461.11
  4723.1  459.74  4788.0  458.58  4841.6  459.50  4894.1  458.95  4910.9  459.02
  4952.5  456.69  4974.4  456.88  4981.7  454.05  4991.7  452.66  4992.5  451.86
  5000.9  452.66  5010.9  455.11  5032.6  456.74  5290.6  457.54  5564.8  461.87
  5601.5  461.61  5691.0  463.06  5713.0  462.48  5863.5  465.38  5997.5  467.61
#Mann=8,-1,0
  3524.4     0.1       0  4723.1    0.05       0  4841.6    0.12       0
  4894.1     0.1       0  4991.7    0.07       0  5000.9     0.1       0
  5601.5    0.05       0  5863.5     0.1       0
Bank Sta=4991.7,5000.9
Exp/Cntr=0.3,0.1

Type RM Length L Ch R = 1,21833,649,649,649
BEGIN DESCRIPTION:
Calf Creek 38.0
END DESCRIPTION:
XS GIS Cut Line= 3
      2006981.52     13450853.48      2007988.45     13449367.39
      2008550.38     13448510.62
#Sta/Elev= 30
  3237.7  467.48  3549.9  460.39  3576.9  458.85  3642.8  458.22  3648.8  459.36
  3663.8  459.28  3879.4  457.15  3924.3  455.00  3936.5  456.70  4053.1  458.01
  4514.4  458.40  4575.5  456.73  4601.5  457.74  4823.0  457.72  4939.0  455.37
  4975.3  456.02  4987.7  454.54  4998.1  451.57  4998.9  450.77  5007.3  451.57
  5017.6  455.92  5023.7  456.15  5155.2  455.43  5191.1  453.63  5234.6  456.29
  5476.0  461.62  5767.1  468.99  5855.5  471.62  5942.9  472.07  6057.4  475.31
#Mann=7,-1,0
  3237.7     0.1       0  4575.5    0.05       0  4601.5     0.1       0
  4998.1    0.07       0  5007.3     0.1       0  5476.0    0.05       0
  5767.1     0.1       0
Bank Sta=4998.1,5007.3
Exp/Cntr=0.3,0.1

Type RM Length L Ch R = 1,21184,726,726,726
BEGIN DESCRIPTION:
Calf Creek 37.0
END DESCRIPTION:
XS GIS Cut Line= 3
      2007675.95     13450829.20      2008425.00     13449475.00
      2008710.19     13448750.57
#Sta/Elev= 30
  3441.2  471.75  3450.6  471.78  3532.0  465.11  3613.3  460.33  3708.8  457.03
  3862.9  453.84  3922.5  454.10  3944.3  453.16  3950.0  454.01  3960.3  452.73
  3982.1  453.89  4106.9  454.49  4200.2  454.58  4241.4  453.52  4275.2  455.34
  4350.6  455.21  4965.9  454.65  4980.7  453.89  4985.9  451.32  4991.4  451.32
  4993.6  450.24  4994.5  449.44  5002.1  449.44  5003.0  450.24  5010.3  453.50
  5302.7  461.63  5353.0  462.94  5496.5  469.29  5594.8  471.75  5767.3  477.08
#Mann=7,-1,0
  3441.2     0.1       0  4241.4    0.08       0  4350.6     0.1       0
  4993.6    0.07       0  5003.0     0.1       0  5302.7    0.05       0
  5594.8     0.1       0
Bank Sta=4993.6,5003
Exp/Cntr=0.3,0.1

Type RM Length L Ch R = 1,20458,462,462,462
BEGIN DESCRIPTION:
Calf Creek 36.0
END DESCRIPTION:
XS GIS Cut Line= 4
      2007775.02     13451024.96      2008262.76     13450106.97
      2008710.68     13449818.78      2008924.99     13449025.04
#Sta/Elev= 30
  3582.3  480.16  3700.3  476.09  3899.3  460.53  3974.7  457.33  4261.7  452.70
  4298.8  453.14  4329.6  450.96  4337.1  452.43  4359.1  452.94  4480.4  453.30
  4507.1  453.34  4950.2  452.03  4986.5  451.42  4993.1  450.41  5002.9  446.35
  5003.8  445.55  5012.3  446.35  5016.9  449.42  5038.0  452.16  5210.1  451.98
  5261.8  453.13  5267.0  454.46  5293.0  453.69  5427.7  458.02  5530.8  460.42
  5552.0  459.62  5570.7  461.25  5616.2  461.87  5897.9  474.52  5976.6  478.42
#Mann=7,-1,0
  3582.3     0.1       0  4480.4    0.05       0  4507.1     0.1       0
  5002.9    0.07       0  5012.3     0.1       0  5616.2    0.05       0
  5897.9     0.1       0
Bank Sta=5002.9,5012.3
Exp/Cntr=0.3,0.1

Type RM Length L Ch R = 1,19996,454,454,454
BEGIN DESCRIPTION:
Calf Creek 35.0
END DESCRIPTION:
XS GIS Cut Line= 3
      2007998.86     13451159.07      2008675.00     13450175.00
      2009275.02     13449374.98
#Sta/Elev= 30
  3854.0  474.65  3983.0  467.72  4156.2  461.86  4551.4  454.76  4728.3  452.75
  4825.4  450.92  4867.3  451.84  4897.1  448.99  4926.6  449.16  4939.0  446.35
  4947.8  449.71  4962.7  449.43  4968.8  445.81  4978.6  445.19  4979.6  444.39
  4988.8  445.19  5004.7  447.03  5011.6  450.26  5034.5  451.94  5069.8  449.98
  5119.8  450.10  5469.8  453.72  5490.7  450.85  5505.3  453.36  5526.1  450.64
  5555.3  453.97  5561.5  452.34  5611.5  452.80  5799.7  460.18  6048.0  468.09
#Mann=6,-1,0
  3854.0     0.1       0  4551.4    0.05       0  4728.3     0.1       0
  4978.6    0.07       0  4988.8     0.1       0  5799.7    0.05       0
Bank Sta=4978.6,4988.8
Exp/Cntr=0.3,0.1

Type RM Length L Ch R = 1,19542,682,682,682
BEGIN DESCRIPTION:
Calf Creek 34.0
END DESCRIPTION:
XS GIS Cut Line= 3
      2008475.01     13451274.97      2008978.04     13450117.39
      2009375.00     13449375.01
#Sta/Elev= 30
  3733.7  474.22  3929.9  468.55  4115.3  458.67  4232.8  454.88  4346.0  453.07
  4638.6  449.22  4660.5  446.52  4682.3  449.64  4867.6  451.19  4973.4  449.33
  4978.9  448.85  4987.6  445.37  4989.3  443.31  4990.3  442.51  4999.5  443.31
  5009.9  448.49  5032.6  450.56  5068.0  449.82  5106.2  446.04  5112.0  447.40
  5180.0  449.59  5215.9  448.91  5270.4  452.05  5292.3  449.68  5314.3  452.41
  5336.2  451.87  5380.1  455.31  5531.8  458.65  5778.2  467.12  5837.7  469.25
#Mann=7,-1,0
  3733.7     0.1       0  4232.8    0.05       0  4346.0     0.1       0
  4989.3    0.07       0  4999.5     0.1       0  5531.8    0.05       0
  5778.2     0.1       0
Bank Sta=4989.3,4999.5
Exp/Cntr=0.3,0.1

Type RM Length L Ch R = 1,18860,357,357,357
BEGIN DESCRIPTION:
Calf Creek 33.0
END DESCRIPTION:
XS GIS Cut Line= 3
      2008625.00     13451175.01      2009365.97     13450047.92
      2009509.30     13449492.35
#Sta/Elev= 30
  3552.9  471.05  3653.8  467.17  3833.4  457.30  3949.1  453.90  4108.8  451.01
  4202.1  447.97  4217.2  449.58  4223.2  447.82  4232.3  447.54  4247.0  448.31
  4268.5  447.19  4274.4  448.17  4289.5  445.61  4295.5  446.73  4310.6  445.89
  4325.7  448.24  4485.4  449.15  4687.2  449.47  4905.8  447.43  4987.4  446.10
  4995.2  443.02  4995.3  441.93  4996.2  441.13  5005.5  441.93  5008.0  445.86
  5018.4  448.19  5049.3  451.62  5175.2  454.56  5427.8  463.59  5475.5  465.45
#Mann=7,-1,0
  3552.9     0.1       0  3833.4    0.05       0  3949.1     0.1       0
  4995.3    0.07       0  5005.5     0.1       0  5175.2    0.05       0
  5427.8     0.1       0
Bank Sta=4995.3,5005.5
Exp/Cntr=0.3,0.1

Type RM Length L Ch R = 1,18503,77,77,77
BEGIN DESCRIPTION:
Mapping XS 5c222f87
END DESCRIPTION:
XS GIS Cut Line= 5
      2008869.97     13451052.00      2009330.92     13450218.65
      2009442.90     13450200.42      2009580.92     13450098.86
      2009859.32     13449539.45
#Sta/Elev= 30
  3855.8  459.94  3866.9  459.33  3977.7  455.75  4343.8  448.03  4372.4  447.13
  4394.1  444.92  4415.9  447.33  4491.5  448.32  4812.7  448.37  4961.8  445.67
  4991.1  444.00  4993.6  442.91  4994.5  442.11  5003.8  442.91  5048.4  447.72
  5070.6  447.84  5076.8  446.65  5085.2  447.68  5108.1  445.86  5130.5  445.74
  5136.1  447.92  5152.9  446.80  5158.5  448.47  5175.3  448.16  5180.8  449.75
  5197.7  450.80  5421.2  454.70  5516.7  461.70  5622.2  466.38  5717.8  473.07
#Mann=5,-1,0
  3855.8     0.1       0  3866.9    0.05       0  3977.7     0.1       0
  4993.6    0.07       0  5003.8     0.1       0
Bank Sta=4993.6,5003.8
Exp/Cntr=0.3,0.1

Type RM Length L Ch R = 1,18426,228,228,228
BEGIN DESCRIPTION:
Calf Creek 32.0
END DESCRIPTION:
XS GIS Cut Line= 5
      2008896.91     13451077.12      2009336.13     13450292.43
      2009429.88     13450285.49      2009660.78     13450146.60
      2009924.99     13449525.03
#Sta/Elev= 30
  3877.3  460.33  3915.8  458.58  3943.9  457.05  3965.6  457.37  4026.9  455.43
  4187.1  451.28  4361.1  448.63  4429.8  446.41  4436.0  444.66  4441.7  444.56
  4464.2  447.17  4495.3  447.83  4663.2  448.59  4810.0  447.78  4845.6  449.26
  4870.6  448.69  4897.3  445.61  4918.7  445.29  4924.5  447.01  4982.8  447.78
  4998.3  445.82  4999.8  439.66  5000.8  438.86  5010.0  439.66  5013.9  440.63
  5019.7  444.39  5056.6  446.51  5196.1  448.09  5471.7  453.36  5815.4  474.52
#Mann=5,-1,0
  3877.3     0.1       0  3915.8    0.05       0  4026.9     0.1       0
  4999.8    0.07       0  5010.0     0.1       0
Bank Sta=4999.8,5010
Exp/Cntr=0.3,0.1

Type RM Length L Ch R = 1,18198,335,335,335
BEGIN DESCRIPTION:
Mapping XS 2ccfbb20
END DESCRIPTION:
XS GIS Cut Line= 4
      2009310.09     13451281.14      2009583.52     13450528.54
      2009833.52     13450096.25      2010002.55     13449589.18
#Sta/Elev= 30
  3993.4  463.90  4228.0  454.83  4253.3  453.09  4283.9  453.02  4401.0  448.79
  4510.6  446.97  4518.1  448.26  4523.4  446.77  4548.7  447.87  4554.0  446.52
  4604.6  446.10  4609.9  445.12  4635.2  445.66  4640.5  444.53  4665.8  445.72
  4696.4  445.21  4721.7  446.39  4805.5  446.77  4891.7  444.02  4972.1  444.83
  4998.5  441.36  4999.4  440.56  5007.7  440.56  5008.7  441.36  5030.9  446.73
  5272.1  447.39  5507.3  451.41  5602.2  456.88  5755.0  467.73  5828.0  471.40
#Mann=3,-1,0
  3993.4     0.1       0  4998.5    0.07       0  5008.7     0.1       0
Bank Sta=4998.5,5008.7
Exp/Cntr=0.3,0.1

Type RM Length L Ch R = 1,17863,556,556,556
BEGIN DESCRIPTION:
Calf Creek 31.0
END DESCRIPTION:
XS GIS Cut Line= 3
      2009432.90     13451339.61      2009804.43     13450631.28
      2010214.14     13449631.31
#Sta/Elev= 30
  4167.1  466.68  4417.1  455.65  4736.7  445.48  4764.4  443.61  4808.5  443.11
  4824.9  441.21  4838.5  441.40  4847.0  443.77  4852.6  442.85  4951.5  442.98
  4985.8  441.73  4999.3  439.32  5000.2  438.52  5008.5  438.52  5009.5  439.32
  5009.8  440.15  5017.0  441.90  5039.2  444.45  5484.9  445.81  5698.5  449.25
  5751.9  451.92  5762.6  451.12  5823.9  456.36  5882.7  459.47  5901.3  461.26
  5906.7  460.79  5913.9  461.66  5936.1  461.68  6032.0  465.25  6047.6  465.05
#Mann=3,-1,0
  4167.1     0.1       0  4999.3    0.07       0  5009.5     0.1       0
Bank Sta=4999.3,5009.5
Exp/Cntr=0.3,0.1

Type RM Length L Ch R = 1,17307,352,352,352
BEGIN DESCRIPTION:
Calf Creek 30.0
END DESCRIPTION:
XS GIS Cut Line= 3
      2009866.91     13451721.59      2010200.26     13451006.28
      2010502.35     13449565.27
#Sta/Elev= 30
  3943.4  465.01  4256.3  457.00  4307.5  456.57  4358.9  454.31  4480.2  452.21
  4601.6  448.06  4917.8  442.76  4958.7  440.30  4979.6  440.32  4994.4  435.96
  4995.3  435.16  5003.7  435.16  5004.7  435.96  5009.7  438.60  5019.3  439.83
  5024.4  439.32  5040.4  440.62  5074.3  438.85  5091.5  442.75  5111.9  443.32
  5479.7  442.68  5657.9  446.81  5757.8  450.29  5802.6  452.77  5908.9  455.88
  5929.3  457.43  6002.2  457.59  6031.5  458.54  6113.2  463.67  6204.9  471.30
#Mann=3,-1,0
  3943.4     0.1       0  4994.4    0.07       0  5004.7     0.1       0
Bank Sta=4994.4,5004.7
Exp/Cntr=0.3,0.1
