--- UNT 022 in RCW.prj (project) ---

Proj Title=UNT 022 in RCW Base Level Engineering
Current Plan=p01
Default Exp/Contr=0.3,0.1
English Units
Geom File=g01
Flow File=f01
Plan File=p01
Y Axis Title=Elevation
X Axis Title(PF)=Main Channel Distance
X Axis Title(XS)=Station
BEGIN DESCRIPTION:
UNT 022 in RCW
END DESCRIPTION:
DSS Export Rating Curves= 0
DSS Export Rating Curve Sorted= 0
DSS Export Volume Flow Curves= 0
DXF OffsetX= 0
DXF OffsetY= 0
DXF ScaleX= 1
DXF ScaleY= 10

--- UNT 022 in RCW.p01 (plan) ---

Plan Title=Multiple Run
Short Identifier=Multiple
Geom File=g01
Flow File=f01
Subcritical Flow
K Sum by GR= 0
Std Step Tol= 0.01
Critical Tol= 0.01
Num of Std Step Trials= 20
Max Error Tol= 0.3
Flow Tol Ratio= 0.001
Split Flow NTrial= 30
Split Flow Tol= 0.02
Split Flow Ratio= 0.02
Log Output Level= 0
Friction Slope Method= 1
Unsteady Friction Slope Method= 2
Unsteady Bridges Friction Slope Method= 1
Parabolic Critical Depth
Global Vel Dist=  1 , 1 , 1
Global Log Level= 0
CheckData=True
Encroach Param= -1, 0, 0, 0
BEGIN DESCRIPTION:
Multiple Run
END DESCRIPTION:

--- UNT 022 in RCW.f01 (steady flow) ---

Flow Title=Multiple
Program Version=5.05
Number of Profiles= 7
Profile Names=10-year,25-year,50-year,1pct_min,100-year,1pct_plu,500-year
River Rch & RM=UNT 022 in RCW,Reach-1         ,41525
     150     205     249     152     303     604     455
River Rch & RM=UNT 022 in RCW,Reach-1         ,40544
     268     377     468     290     578    1154     899
River Rch & RM=UNT 022 in RCW,Reach-1         ,33487
     372     531     666     416     830    1657    1313
River Rch & RM=UNT 022 in RCW,Reach-1         ,31702
     406     581     730     457     912    1821    1448
River Rch & RM=UNT 022 in RCW,Reach-1         ,28589
     553     801    1015     640    1276    2547    2052
River Rch & RM=UNT 022 in RCW,Reach-1         ,23769
     598     867    1099     693    1382    2758    2224
River Rch & RM=UNT 022 in RCW,Reach-1         ,20168
     615     890    1127     709    1415    2824    2269
River Rch & RM=UNT 022 in RCW,Reach-1         ,16599
     608     876    1105     693    1383    2759    2201
River Rch & RM=UNT 022 in RCW,Reach-1         ,12421
     640     921    1160     726    1449    2891    2298
River Rch & RM=UNT 022 in RCW,Reach-1         ,7278
     665     957    1207     756    1508    3009    2396
River Rch & RM=UNT 022 in RCW,Reach-1         ,5214
    1192    1755    2246    1426    2846    5679    4644
River Rch & RM=UNT 022 in RCW,Reach-1         ,234
    1228    1809    2319    1474    2942    5869    4810
Boundary for River Rch & Prof#=UNT 022 in RCW,Reach-1         , 1
Up Type= 0
Dn Type= 3
Dn Slope=0.01356
Boundary for River Rch & Prof#=UNT 022 in RCW,Reach-1         , 2
Up Type= 0
Dn Type= 3
Dn Slope=0.01356
Boundary for River Rch & Prof#=UNT 022 in RCW,Reach-1         , 3
Up Type= 0
Dn Type= 3
Dn Slope=0.01356
Boundary for River Rch & Prof#=UNT 022 in RCW,Reach-1         , 4
Up Type= 0
Dn Type= 3
Dn Slope=0.01356
Boundary for River Rch & Prof#=UNT 022 in RCW,Reach-1         , 5
Up Type= 0
Dn Type= 3
Dn Slope=0.01356
Boundary for River Rch & Prof#=UNT 022 in RCW,Reach-1         , 6
Up Type= 0
Dn Type= 3
Dn Slope=0.01356
Boundary for River Rch & Prof#=UNT 022 in RCW,Reach-1         , 7
Up Type= 0
Dn Type= 3
Dn Slope=0.01356
DSS Import GetInterval= 0
DSS Import GetPeak= 0
DSS Import FillOption= 0

--- UNT 022 in RCW.g01 (geometry) ---

Geom Title=Existing Conditions
Program Version=5.05

River Reach=UNT 022 in RCW  ,Reach-1
Reach XY= 30
       1970250.8     13474354.54       1971740.8     13473924.54
       1972560.8     13473994.54       1973710.8     13473464.54
       1974280.8     13473894.54       1975851.9     13474138.93
      1976326.74     13474386.17      1976566.89     13475531.52
       1978170.8     13476404.54       1979810.8     13476184.54
       1980890.8     13476494.54       1981580.8     13476344.54
      1983085.74     13475543.95      1983778.45     13474483.53
      1984951.89     13473557.83      1986176.04     13471855.97
      1987020.23     13471553.24       1987480.8     13469504.54
       1987110.8     13468074.54       1987260.8     13467514.54
       1987790.8     13466804.54       1988210.8     13466624.54
       1989070.8     13465754.54       1990910.8     13465394.54
      1992120.16      13463490.8       1993660.8     13462334.54
      1994052.49     13461416.79      1995447.89     13460699.56
      1996405.86     13460853.85       1999330.8     13459764.54

Type RM Length L Ch R = 1 ,41525   ,471,471,471
BEGIN DESCRIPTION:
UNT 022 in RCW 81.0
END DESCRIPTION:
XS GIS Cut Line= 3
      1971024.97     13474874.97        1970475.       13474325.
      1970181.27     13473766.06
#Sta/Elev= 30
  4221.7  605.06  4306.5  603.36  4348.9  601.94  4447.9  595.94  4504.5  593.11
  4603.5  589.33  4688.4  587.14  4759.1  587.12  4812.6  586.08  4813.1  585.28
  4818.1  585.28  4818.6  586.08  4914.6  587.19    4982   586.6  5013.3  586.68
  5089.9  589.39    5184  594.14  5250.2  598.92  5266.6  601.05  5354.7  608.36
  5371.1  608.64    5465  613.54  5481.4  613.88  5525.5   616.2  5531.1  617.01
  5563.9  617.15  5569.6  617.83  5585.9  617.48  5613.6  618.59  5630.9  617.85
#Mann= 4 ,-1 , 0
  4221.7     .05       0  4812.6     .07       0  4818.6     .05       0
    4982      .1       0
Bank Sta=4812.6,4818.6
XS Rating Curve= 0 ,0
Exp/Cntr=0.3,0.1

Type RM Length L Ch R = 1 ,41054   ,510,510,510
BEGIN DESCRIPTION:
UNT 022 in RCW 80.0
END DESCRIPTION:
XS GIS Cut Line= 3
      1971384.39     13474930.11        1970875.       13474175.
      1970329.85     13473635.98
#Sta/Elev= 30
    4129  605.94  4255.8  605.12  4492.7  599.14  4528.7  598.36  4557.4  598.57
  4600.7   595.1  4702.1  590.01  4822.7  585.72  4900.4   584.2  4900.9   583.4
  4905.9   583.4  4906.4   584.2  4945.5  584.81  5061.1  584.51  5167.1  586.74
  5187.8   588.1  5336.8  593.32  5358.1  594.83  5407.5  596.06  5442.9  597.85
    5450  597.59  5499.5   600.1  5534.8  600.94  5556.1  602.29  5697.5  606.26
  5718.7  606.25  5768.2  608.41  5775.2  607.95  5803.5  609.67  5806.5  610.33
#Mann= 4 ,-1 , 0
    4129     .05       0  4900.4    .035       0  4906.4     .05       0
  5187.8      .1       0
Bank Sta=4900.4,4906.4
XS Rating Curve= 0 ,0
Exp/Cntr=0.3,0.1

Type RM Length L Ch R = 1 ,40544   ,362,362,362
BEGIN DESCRIPTION:
UNT 022 in RCW 79.0
END DESCRIPTION:
XS GIS Cut Line= 3
      1971920.86     13474904.09        1971225.       13473975.
      1970712.55     13473385.88
#Sta/Elev= 30
  4035.9  606.34  4039.2  605.68  4068.3  605.26    4110  602.41    4233  597.41
  4253.8  595.99    4383  591.39  4403.8  590.35  4410.1  589.48  4418.4  589.25
    4433  590.03  4439.2  591.22  4455.5  590.91    4533  589.63  4589.3  590.31
  4639.3  589.82  4753.9  586.61 4930.81583.3935  5036.4   582.4  5036.9   581.6
  5041.9   581.6  5042.4   582.4  5203.8  582.66 5260.96583.3934  5451.6  587.27
  5678.6  594.48  5848.5  601.73  5912.4  605.17  5932.4  607.11  5977.5  610.32
#Mann= 5 ,-1 , 0
  4035.9      .1       0  4455.5     .05       0  5036.4    .035       0
  5042.4     .05       0  5932.4      .1       0
Bank Sta=4930.81,5260.96
XS Rating Curve= 0 ,0
Exp/Cntr=0.3,0.1

Type RM Length L Ch R = 1 ,40182   ,388,388,388
BEGIN DESCRIPTION:
UNT 022 in RCW 78.0
END DESCRIPTION:
XS GIS Cut Line= 3
      1971928.68     13474648.89        1971575.       13473825.
      1971056.27     13473115.01
#Sta/Elev= 30
  4290.2   599.7  4305.3  599.16  4316.9  597.89    4335  597.65  4370.6  595.19
  4416.6  593.53  4446.8   591.3  4457.7  591.79  4492.7  588.88  4539.8  586.97
  4615.9  584.93  4697.8  583.77  4899.8581.5351  5009.7  580.49  5010.2  579.69
  5015.2  579.69  5015.7  580.49  5101.6  581.44 5223.74581.5351  5309.2  582.16
  5486.8   587.1  5566.4  588.11  5622.8  589.94  5681.4  590.72  5773.3  593.18
  5838.2  593.78  5873.7  595.07  5974.1  594.91  6009.7  595.72  6066.1  595.74
#Mann= 4 ,-1 , 0
  4290.2      .1       0  4697.8     .05       0  5009.7    .035       0
  5015.7     .05       0
Bank Sta=4899.8,5223.74
XS Rating Curve= 0 ,0
Exp/Cntr=0.3,0.1

Type RM Length L Ch R = 1 ,39794   ,542,542,542
BEGIN DESCRIPTION:
UNT 022 in RCW 77.0
END DESCRIPTION:
XS GIS Cut Line= 3
        1972075.     13474574.97        1971975.       13473975.
      1971913.04     13473255.61
#Sta/Elev= 30
  4396.3  600.63  4467.2  597.76  4545.8  592.06  4558.5  591.59  4568.6  592.31
  4578.8  591.29  4639.6  588.71  4689.2  585.77  4789.1  581.85 4879.72579.6887
    4964  578.68  4968.5  578.16    4969  577.36  4974.2  577.36  4974.7  578.16
  5014.6  578.16  5044.7   579.3  5091.5  579.55    5115  580.04    5125  579.56
 5218.37579.6887  5245.4  580.84  5275.5  580.71  5311.9  582.36    5396  586.12
  5486.3  589.21  5530.2  589.92  5586.7  592.54  5643.7   593.8  5726.6  593.84
#Mann= 6 ,-1 , 0
  4396.3      .1       0  4689.2     .05       0  4968.5    .035       0
  4974.7     .05       0  5091.5      .1       0  5311.9     .05       0
Bank Sta=4879.72,5218.37
XS Rating Curve= 0 ,0
Exp/Cntr=0.3,0.1

Type RM Length L Ch R = 1 ,39252   ,653,653,653
BEGIN DESCRIPTION:
UNT 022 in RCW 76.0
END DESCRIPTION:
XS GIS Cut Line= 3
      1972814.08     13474940.52      1972405.23     13473695.74
      1971998.98     13473247.83
#Sta/Elev= 30
  4004.3  614.53  4041.7   612.3  4048.2   611.2  4094.3  607.78    4168  605.52
  4283.8  599.45  4294.3  599.82  4315.4  598.13  4403.4  594.53  4452.2  591.37
  4473.2  592.16  4504.8   589.4  4538.3  588.08  4753.3  580.09  4890.7577.1617
    4941  576.28  4941.5  575.48  4946.8  575.48  4947.3  576.28  5263.2  577.54
  5283.7   578.3 5329.25 577.162  5421.6  578.63  5473.1   580.3    5577  584.51
    5648  586.46  5739.9  590.76  5782.5  591.03  5831.8  592.63  5919.2  592.91
#Mann= 6 ,-1 , 0
  4004.3      .1       0  4538.3     .05       0    4941    .035       0
  4947.3     .05       0  5263.2      .1       0  5473.1     .05       0
Bank Sta=4890.7,5329.25
XS Rating Curve= 0 ,0
Exp/Cntr=0.3,0.1

Type RM Length L Ch R = 1 ,38599   ,332,332,332
BEGIN DESCRIPTION:
UNT 022 in RCW 75.0
END DESCRIPTION:
XS GIS Cut Line= 4
      1973110.96     13474615.02      1973181.27     13473943.13
      1972801.06     13473486.88      1972051.06     13473036.89
#Sta/Elev= 30
  4154.7  596.01  4295.5  590.99    4396   585.1  4406.1  585.54  4466.4  583.08
    4567  581.05  4617.2  580.33  4629.1  581.13  4647.4  580.27  4677.6  576.24
  4687.6  576.11  4707.7  579.15  4798.2  576.11  4834.7  575.89 4886.64574.8617
  5014.9  573.48  5015.4  572.68  5020.8  572.68  5021.3  573.48  5244.6  575.09
 5387.73574.8618  5495.6  575.92  5808.5  575.77  5962.1  579.82  6063.2  581.28
  6078.7  582.42  6142.8  583.51  6173.9   585.5  6201.2  584.78  6298.8  587.17
#Mann= 4 ,-1 , 0
  4154.7      .1       0  4834.7     .05       0  5014.9    .035       0
  5021.3     .05       0
Bank Sta=4886.64,5387.73
XS Rating Curve= 0 ,0
Exp/Cntr=0.3,0.1

Type RM Length L Ch R = 1 ,38267   ,127,127,127
BEGIN DESCRIPTION:
UNT 022 in RCW 74.0
END DESCRIPTION:
XS GIS Cut Line= 3
      1973248.98     13474461.36      1973397.42     13473693.13
      1972363.57     13472643.67
#Sta/Elev= 30
  4023.2   586.9  4083.5  586.97  4233.4  582.47  4238.9  581.38    4244  582.09
  4263.9  580.25  4284.3  581.62  4342.6  579.42  4426.9  578.53  4518.6  578.39
  4658.6  581.05  4732.4   580.3  4752.8   579.2  4773.2  575.58  4804.6  573.79
 4826.06573.3451  4986.7   572.5  4987.2   571.7  4993.1   572.5  5053.6  573.63
 5373.79 573.345  5619.2  574.82    5796  580.45  5909.2  582.64  6008.2  583.36
  6029.3  582.06  6114.2  582.66  6121.3  583.87  6149.6  584.25  6278.8  584.69
#Mann= 4 ,-1 , 0
  4023.2      .1       0  4804.6     .05       0  4986.7     .04       0
  4993.1     .05       0
Bank Sta=4826.06,5373.79
XS Rating Curve= 0 ,0
Exp/Cntr=0.3,0.1

Type RM Length L Ch R = 1 ,38140   ,229,229,229
BEGIN DESCRIPTION:
Mapping XS 4a427f9a
END DESCRIPTION:
XS GIS Cut Line= 3
      1973282.83     13474424.93      1973519.81     13473641.05
      1972480.72     13472586.34
#Sta/Elev= 30
  3968.9  587.34  4131.3  581.88  4250.9  579.72  4268.3  578.41  4306.5  579.08
  4365.8  577.35  4438.3  577.37  4595.6  579.44  4637.4  577.83  4660.4  574.47
  4684.6  574.07  4689.8  572.58  4717.6  571.08  4722.8  572.71  4755.7  570.55
 4871.16569.4903  4926.7   568.5  4927.2   567.7  4932.6   567.7  4933.1   568.5
 5067.44569.4904  5615.8  574.01  5721.9  576.95  5792.6   580.4  5813.8  580.17
  5856.2  583.47  5912.8  585.53  6018.8  585.85  6110.8  587.89  6268.4  588.98
#Mann= 4 ,-1 , 0
  3968.9      .1       0  4660.4     .05       0  4926.7     .04       0
  4933.1     .05       0
Bank Sta=4871.16,5067.44
XS Rating Curve= 0 ,0
Exp/Cntr=0.3,0.1

Type RM Length L Ch R = 1 ,37911   ,456,456,456
BEGIN DESCRIPTION:
UNT 022 in RCW 73.0
END DESCRIPTION:
XS GIS Cut Line= 3
      1973324.51     13474424.86      1973579.71     13473682.72
      1973673.44     13472419.88
#Sta/Elev= 30
  3993.7  586.82  4197.4  581.43  4223.4   579.7  4342.5  578.13  4416.5  576.15
  4448.3   575.7    4468  576.35  4504.5   575.5  4530.5  576.31  4535.8  575.72
  4647.5  575.95  4655.4  575.53  4670.3  572.73  4680.9  571.76    4692  571.57
  4702.1  572.75  4723.2  570.38  4749.1  569.65 4926.11568.4756  5003.6  567.08
  5004.1  566.28  5009.5  566.28    5010  567.08  5052.3  568.27  5137.2  567.31
 5216.49568.4755  5548.3  574.22  5718.8  578.49  5869.2  583.33  6044.8  585.91
#Mann= 4 ,-1 , 0
  3993.7      .1       0  4647.5     .05       0  5003.6    .035       0
    5010     .05       0
Bank Sta=4926.11,5216.49
XS Rating Curve= 0 ,0
Exp/Cntr=0.3,0.1

Type RM Length L Ch R = 1 ,37455   ,503,503,503
BEGIN DESCRIPTION:
UNT 022 in RCW 72.0
END DESCRIPTION:
XS GIS Cut Line= 3
      1973413.03     13474461.38      1974040.64     13473565.53
      1974038.04     13472721.75
#Sta/Elev= 30
  4063.7  587.22  4133.4  585.03    4163  585.08  4242.4   582.9  4270.2  582.98
  4299.9  581.71  4407.1  579.46  4421.9  578.29  4472.5  577.13  4572.1  573.26
  4600.7  572.89  4615.5  571.92  4627.3  572.44  4636.4  572.26    4646  571.14
    4666  571.04  4701.8   568.6  4758.4  567.41 4909.95565.8632  4984.5  564.83
    4985  564.03  4990.4  564.03  4990.9  564.83  5133.3  566.65    5318  565.44
 5338.24565.8633    5558  569.28    5688  572.04  5838.1  577.14  6001.3  584.76
#Mann= 5 ,-1 , 0
  4063.7      .1       0  4627.3     .08       0    4646     .05       0
  4984.5    .035       0  4990.9     .05       0
Bank Sta=4909.95,5338.24
XS Rating Curve= 0 ,0
Exp/Cntr=0.3,0.1

Type RM Length L Ch R = 1 ,36952   ,386,386,386
BEGIN DESCRIPTION:
UNT 022 in RCW 71.0
END DESCRIPTION:
XS GIS Cut Line= 3
      1974720.32     13474682.69      1974384.39      13474047.3
      1974254.24     13472589.53
#Sta/Elev= 30
  4127.9  580.51  4212.1  578.23  4234.2  577.34  4249.7  575.91  4256.2  576.09
  4261.8  577.54  4272.3  577.35  4283.8  575.75  4322.2  573.11  4382.6  570.03
  4536.6  564.78 4616.58563.3831  4679.4  562.48  4736.1  562.54  4767.4  563.34
    4804  562.77  4889.1  563.06  4946.1  562.16  4946.6  561.36    4952  561.36
  4952.5  562.16 5066.97563.3832  5320.8   565.3  5491.5  564.67  5796.7  570.57
  6063.8  578.08  6164.2  582.35  6224.4  583.94  6242.4  585.39  6310.2  588.49
#Mann= 3 ,-1 , 0
  4127.9     .05       0  4946.1    .035       0  4952.5     .05       0
Bank Sta=4616.58,5066.97
XS Rating Curve= 0 ,0
Exp/Cntr=0.3,0.1

Type RM Length L Ch R = 1 ,36566   ,105,105,105
BEGIN DESCRIPTION:
UNT 022 in RCW 70.0
END DESCRIPTION:
XS GIS Cut Line= 3
      1974689.08     13474523.88        1974725.       13473925.
      1974819.22     13472628.97
#Sta/Elev= 30
  4412.7  577.46  4427.3   575.5  4432.3  576.07  4461.7  574.28  4551.8  569.85
  4732.1  563.33 4771.22562.2479  4822.3  561.27  4842.3  561.55  4849.2  561.23
  4849.7  560.43  4855.1  560.43  4855.6  561.23  5042.7  562.05  5062.8  561.74
 5110.59562.2477  5333.5   563.6  5393.7  562.83  5463.8  563.01  5564.1  563.82
  5631.3  564.83  5636.3   564.6  5664.4   565.2  5724.5  565.64    5895  568.93
  5909.5  568.79  5985.2  570.19  6105.5  571.55  6215.8  574.37  6312.1  575.77
#Mann= 3 ,-1 , 0
  4412.7     .05       0  4849.2    .035       0  4855.6     .05       0
Bank Sta=4771.22,5110.59
XS Rating Curve= 0 ,0
Exp/Cntr=0.3,0.1

Type RM Length L Ch R = 1 ,36461   ,144,144,144
BEGIN DESCRIPTION:
Mapping XS ece8405d
END DESCRIPTION:
XS GIS Cut Line= 4
      1974718.76       13474423.       1974788.2     13474013.28
      1975229.18     13473370.92      1975354.17     13472641.77
#Sta/Elev= 30
  4522.9  572.63  4528.1  572.02  4533.2  572.39  4588.5  569.41  4593.6  569.78
  4648.8  567.09  4653.9  567.33  4769.5  562.78  4774.6  562.97 4808.93561.8844
  4842.2  561.08  4842.7  560.28  4848.1  560.28  4848.6  561.08  4948.5  561.43
  5049.6  561.26  5166.1  561.97  5201.9  561.73    5208  562.09  5360.3  561.44
  5467.9  561.74  5530.8  561.42 5615.98561.8844  5725.6     562    5886  563.19
  6058.4  567.46    6099  568.02  6230.9  571.26  6315.7  572.63  6457.4  573.49
#Mann= 3 ,-1 , 0
  4522.9     .05       0  4842.2    .035       0  4848.6     .05       0
Bank Sta=4808.93,5615.98
XS Rating Curve= 0 ,0
Exp/Cntr=0.3,0.1

Type RM Length L Ch R = 1 ,36317   ,146,146,146
BEGIN DESCRIPTION:
Mapping XS e078664e
END DESCRIPTION:
XS GIS Cut Line= 4
      1974729.15     13474426.52      1974868.06      13474148.7
      1975465.29     13473291.06      1975548.33      13472758.2
#Sta/Elev= 30
  4567.7  572.96  4572.3  573.44  4589.1  572.21  4594.7  572.63  4611.4  571.56
    4617  572.03  4656.1  570.28  4661.7  570.55  4706.5  569.29  4723.2  567.86
  4728.8  568.06  4745.6  566.79  4751.2  566.96  4767.9   565.6 4906.75561.4159
  4929.8  560.78  5004.2  560.63  5004.7  559.83  5010.3  559.83  5010.8  560.63
    5052  561.23  5201.2  561.56  5323.4  560.87  5582.6  561.28  5662.7  560.75
 5855.09561.4159  5949.4  561.69  6030.7  563.03    6385  573.56  6462.7  573.97
#Mann= 3 ,-1 , 0
  4567.7     .05       0  5004.2    .035       0  5010.8     .05       0
Bank Sta=4906.75,5855.09
XS Rating Curve= 0 ,0
Exp/Cntr=0.3,0.1

Type RM Length L Ch R = 1 ,36171   ,140,140,140
BEGIN DESCRIPTION:
Mapping XS 9a9c190b
END DESCRIPTION:
XS GIS Cut Line= 4
      1974709.91      13474479.6      1975220.33     13473935.32
      1975788.04      13473359.8      1976066.69     13472773.86
#Sta/Elev= 30
  4472.1  574.51  4535.4  574.75  4542.7  573.82    4677  572.12  4818.7  565.49
    4995560.5057  5409.4  559.85  5409.9  559.05  5416.2  559.85  5476.4  561.14
  5511.8  560.06  5660.2  560.98  5801.6  560.35    5837  560.84  5844.1  562.45
  5865.2  560.19 6058.71560.5059  6244.4   561.7  6390.8  566.48  6397.4  567.11
  6403.4  569.79  6408.9   567.8  6426.1  571.87  6431.6  570.33  6448.8  572.02
  6454.3  570.19  6471.5   571.3  6477.1  569.26  6582.6  570.32  6675.5  571.08
#Mann= 5 ,-1 , 0
  4472.1     .05       0  5409.4    .035       0  5416.2     .05       0
  6390.8      .1       0  6582.6     .05       0
Bank Sta=4995,6058.71
XS Rating Curve= 0 ,0
Exp/Cntr=0.3,0.1

Type RM Length L Ch R = 1 ,36031   ,335,335,335
BEGIN DESCRIPTION:
UNT 022 in RCW 69.0
END DESCRIPTION:
XS GIS Cut Line= 3
      1974770.66     13474537.34      1975879.62     13473400.17
      1976174.76     13472770.82
#Sta/Elev= 30
  4381.5  579.35  4527.6  577.77  4619.6  573.71  4654.9  573.08    4747  567.59
  4888.2  560.99    4959  559.18  5023.4   558.9  5065.6  558.28 5071.89558.1445
  5168.9  557.87  5199.2  557.75  5314.4   558.3  5377.8  558.31  5489.3  557.44
  5538.9  557.77  5545.9  558.59  5553.1  557.67  5772.2  558.13  5867.9  557.03
  5868.4  556.23  5874.2  556.23  5874.7  557.03 5987.61558.1445  6135.7  560.35
  6204.2  562.75    6301  564.26  6460.7  568.78  6616.2  571.38    6665  571.46
#Mann= 9 ,-1 , 0
  4381.5     .05       0  5023.4      .1       0  5065.6     .05       0
  5168.9      .1       0  5199.2     .05       0  5314.4      .1       0
  5377.8     .05       0  5867.9     .04       0  5874.7     .05       0
Bank Sta=5071.89,5987.61
XS Rating Curve= 0 ,0
Exp/Cntr=0.3,0.1

Type RM Length L Ch R = 1 ,35696   ,251,251,251
BEGIN DESCRIPTION:
UNT 022 in RCW 68.0
END DESCRIPTION:
XS GIS Cut Line= 3
      1975094.29     13474724.13        1975525.       13474125.
      1976215.99     13472762.15
#Sta/Elev= 30
  4261.6  574.38  4340.2  574.01    4355  574.49  4375.9  573.77  4390.6  574.27
  4526.8  572.08  4618.9  569.48  4698.7     566  4957.3  557.24  4967.8  557.13
  5013.4  556.27  5287.6  556.11  5288.1  555.31  5293.9  555.31  5294.4  556.11
  5347.4   556.8  5581.2   557.3  5603.5     558  5662.7  556.78 5738.73557.1298
  5974.9  560.14  6026.6  562.17  6109.5  563.45  6255.2  567.23  6293.8   567.5
  6310.4  568.57  6389.8  569.37  6434.6  570.84  6471.9  570.86  6527.5  572.06
#Mann= 5 ,-1 , 0
  4261.6     .05       0  4957.3      .1       0  5287.6     .07       0
  5294.4      .1       0  5662.7     .05       0
Bank Sta=4967.8,5738.73
XS Rating Curve= 0 ,0
Exp/Cntr=0.3,0.1

Type RM Length L Ch R = 1 ,35445   ,242,242,242
BEGIN DESCRIPTION:
Mapping XS 84c80bcc
END DESCRIPTION:
XS GIS Cut Line= 3
      1975382.49     13474547.04      1975983.21      13473873.4
      1976969.32     13472890.77
#Sta/Elev= 30
  4427.9  570.46    4516  571.24  4636.4  570.17    4700     567  4721.7  564.63
  4728.4  564.95  4735.9  563.66  4785.2   560.9  4799.4  559.43 4922.97555.6691
  5040.2  555.08  5096.9  555.44  5260.1  555.86  5383.8  554.49  5384.3  553.69
  5390.1  553.69  5390.6  554.49 5518.32555.6691  5648.8  556.39  5747.8  555.84
  5875.1  557.18  5981.2  558.78    6066  562.56  6102.4  563.01    6165  563.75
  6200.4  565.57  6242.8  565.87    6462  571.82  6617.6  573.95  6722.6  573.32
#Mann= 5 ,-1 , 0
  4427.9     .05       0  5096.9      .1       0  5383.8    .035       0
  5390.6      .1       0  6102.4     .05       0
Bank Sta=4922.97,5518.32
XS Rating Curve= 0 ,0
Exp/Cntr=0.3,0.1

Type RM Length L Ch R = 1 ,35203   ,450,450,450
BEGIN DESCRIPTION:
UNT 022 in RCW 67.0
END DESCRIPTION:
XS GIS Cut Line= 3
       1974688.1     13475112.96        1975975.       13474225.
      1977174.99     13473725.01
#Sta/Elev= 30
  3434.2  581.42  3473.8  580.49  3479.9   580.8  3488.7  583.44  3494.7  580.42
  3509.6  579.16  3545.5   580.6  3551.9  579.11  3596.2  576.75  4178.3  567.98
  4306.7  568.85    4423  567.76  4566.4  569.51    4638  568.43  4673.9  567.05
  4739.4  559.87 4867.39555.0342  5248.7  554.27  5298.2  553.35  5298.7  552.55
    5305  553.35 5393.38555.0344  5619.7  560.05  5999.3  566.21  6046.9  568.99
  6070.2  568.48    6146  571.18  6158.5  570.59  6192.6  572.69  6297.7  573.68
#Mann= 6 ,-1 , 0
  3434.2     .05       0  5248.7      .1       0  5298.2    .035       0
    5305      .1       0  5619.7      .1       0  6192.6     .05       0
Bank Sta=4867.39,5393.38
XS Rating Curve= 0 ,0
Exp/Cntr=0.3,0.1

Type RM Length L Ch R = 1 ,34753   ,517,517,517
BEGIN DESCRIPTION:
UNT 022 in RCW 66.0
END DESCRIPTION:
XS GIS Cut Line= 3
      1974858.23     13475380.33        1976375.       13474425.
      1976899.89     13474217.14
#Sta/Elev= 30
  3232.8  570.88  3291.8  570.36  3307.1  569.46    3313  570.06  3364.8  569.52
  3380.1  568.31  3407.2  568.56  3453.1  566.47  3465.3  566.68  3480.2  565.59
  3509.1  564.98  4039.4  556.67 4366.95553.4074  4513.7  552.77  4514.2  551.97
  4520.1  551.97  4520.6  552.77  4871.7  553.69  4975.3  552.95 5018.33553.4075
  5148.3  556.66  5186.7  560.12    5197  561.35  5208.2   563.6  5232.1  566.49
  5256.4  567.81  5346.5  569.01  5394.2  569.04  5455.6  570.75  5589.9  570.72
#Mann= 5 ,-1 , 0
  3232.8      .1       0  3509.1     .05       0  4513.7    .035       0
  4520.6     .05       0  5346.5      .1       0
Bank Sta=4366.95,5018.33
XS Rating Curve= 0 ,0
Exp/Cntr=0.3,0.1

Type RM Length L Ch R = 1 ,34236   ,130,130,130
BEGIN DESCRIPTION:
UNT 022 in RCW 65.0
END DESCRIPTION:
XS GIS Cut Line= 3
      1975490.16     13475713.67      1976691.54      13474748.4
       1977041.1     13474274.25
#Sta/Elev= 30
  3767.7  583.16  3776.9  582.33  3820.1  581.73  3826.5  580.69  3876.1  579.75
  3898.5  579.74  3927.3  578.34  3968.9  574.79  4012.1  572.67  4047.3  569.83
  4253.7  560.75  4268.1  560.71  4317.7  557.54 4469.72552.5836  4538.5  551.26
  4669.5  551.08    4670  550.28    4676  550.28  4676.5  551.08  4901.7  552.59
  5007.4  551.78 5072.12552.5837  5199.4  554.67  5308.8  558.11  5406.8  559.55
  5456.9  561.01  5477.8  562.75  5577.7  565.38    5814  573.38  5897.9  574.16
#Mann= 5 ,-1 , 0
  3767.7      .1       0  3876.1     .05       0  4669.5    .035       0
  4676.5     .05       0  5577.7      .1       0
Bank Sta=4469.72,5072.12
XS Rating Curve= 0 ,0
Exp/Cntr=0.3,0.1

Type RM Length L Ch R = 1 ,34106   ,206,206,206
BEGIN DESCRIPTION:
Mapping XS 874da016
END DESCRIPTION:
XS GIS Cut Line= 4
      1975583.91     13475737.98      1975861.68     13475592.15
      1976875.57     13474692.85      1977132.52     13474300.47
#Sta/Elev= 30
  3900.9  584.45  4006.8  579.83  4045.2  579.11  4139.3  572.42  4171.9  572.13
  4177.5  570.62  4184.5  571.22  4285.9  566.72  4356.5  562.26  4378.2  562.48
  4384.9  561.36  4470.2  558.28  4519.5  554.95  4533.8  555.36  4540.4  554.42
 4605.19 552.519  4742.7  550.71  4743.2  549.91  4749.2  549.91  4749.7  550.71
    5008  551.34 5068.76552.5188  5242.1  555.71  5468.8  562.26  5489.7  561.57
  5597.1  565.63  5637.4  566.45  5741.4  568.49  5958.5  575.42  6038.9   575.8
#Mann= 5 ,-1 , 0
  3900.9      .1       0  4742.7     .07       0  4749.7      .1       0
  5597.1     .05       0  5637.4      .1       0
Bank Sta=4605.19,5068.76
XS Rating Curve= 0 ,0
Exp/Cntr=0.3,0.1

Type RM Length L Ch R = 1 ,33900   ,413,413,413
BEGIN DESCRIPTION:
UNT 022 in RCW 64.0
END DESCRIPTION:
XS GIS Cut Line= 3
      1975840.87     13475762.27        1976475.       13475275.
      1976824.97     13475075.01
#Sta/Elev= 30
  4199.2     583  4206.8  582.06  4242.2  581.76  4300.2  579.68    4350  575.47
  4356.3  574.34  4414.4  571.98  4514.1  565.26  4549.4  562.02  4663.6     556
  4721.5  553.81  4734.3  552.61 4754.65552.3544  4821.3  550.59  4977.1  551.14
  4991.7  551.06  4992.3  550.38  4992.8  549.58  4998.8  549.58  4999.3  550.38
  5028.4  551.51  5093.2  550.94 5152.93552.3547  5227.1  555.58  5248.7  557.95
  5291.9  560.61  5321.4  563.61  5350.9  568.58    5379  570.65    5402  571.07
#Mann= 3 ,-1 , 0
  4199.2      .1       0  4992.3     .07       0  4999.3      .1       0
Bank Sta=4754.65,5152.93
XS Rating Curve= 0 ,0
Exp/Cntr=0.3,0.1

Type RM Length L Ch R = 1 ,33487   ,445,445,445
BEGIN DESCRIPTION:
UNT 022 in RCW 63.0
END DESCRIPTION:
XS GIS Cut Line= 3
      1976174.19     13476043.53        1976675.       13475625.
        1976825.     13475124.98
#Sta/Elev= 30
  4323.4  579.41  4393.7  580.61  4436.6  579.66  4471.8  577.31  4592.8  572.24
  4642.3  565.96  4685.2  563.13    4706  559.81  4720.4  558.63  4755.5  556.41
  4763.3  556.77  4769.8   555.4  4784.1  554.57 4849.56552.1555    4926  549.68
  4986.5  549.88  4994.3  548.78  4994.8  547.98  5000.9  547.98  5001.4  548.78
  5030.9  550.27  5195.3  549.83 5234.77552.1551  5272.7  553.85  5305.8   557.8
  5404.1  562.85  5410.2  563.94  5435.4  564.74  5456.3  567.62  5498.1  569.57
#Mann= 3 ,-1 , 0
  4323.4      .1       0  4994.3     .07       0  5001.4      .1       0
Bank Sta=4849.56,5234.77
XS Rating Curve= 0 ,0
Exp/Cntr=0.3,0.1

Type RM Length L Ch R = 1 ,33042   ,283,283,283
BEGIN DESCRIPTION:
UNT 022 in RCW 62.0
END DESCRIPTION:
XS GIS Cut Line= 3
      1976288.74     13476170.28        1977025.       13475825.
      1977585.67     13475250.98
#Sta/Elev= 30
  4161.1  570.98  4184.9  571.89  4190.5  572.98  4258.9  574.72  4327.4  574.68
  4395.9  572.91  4418.7  571.82    4447  568.42  4532.5  562.34  4566.7  558.94
 4726.36552.1024  4840.5   549.1  4930.1  548.27  4981.4  548.81  4988.4   548.6
  5006.1  545.64  5006.6  544.84  5012.7  544.84  5013.3  545.64  5023.8  548.59
  5115.7  548.26  5193.5  549.74 5244.93552.1025  5363.3  555.17  5370.3  556.23
  5398.6     557  5405.7  556.32    5434  557.52  5660.2  560.93  5776.7  567.23
#Mann= 3 ,-1 , 0
  4161.1      .1       0  5006.1     .07       0  5013.3      .1       0
Bank Sta=4726.36,5244.93
XS Rating Curve= 0 ,0
Exp/Cntr=0.3,0.1

Type RM Length L Ch R = 1 ,32759   ,61,61,61
BEGIN DESCRIPTION:
Mapping XS 1bd3e7a7
END DESCRIPTION:
XS GIS Cut Line= 6
      1976593.47     13476933.26      1976760.12     13476568.71
      1977020.53     13476232.78      1977189.81     13476107.78
      1977296.58     13475860.38      1977537.99     13475328.24
#Sta/Elev= 30
  3820.3  560.26    3956  559.54  4007.6  560.57  4145.7  554.02 4329.78 552.101
  4419.4  552.23    4623  549.28  4689.9  548.85  4733.8  549.81  4783.9  546.31
  4790.1  545.08  4843.5  545.09  4921.4   544.9  4921.9   544.1    4928   544.1
  4928.6   544.9  4997.6  545.16  5094.2  545.12  5126.1  545.65  5142.9  548.26
 5207.81552.1013  5228.2  555.72  5233.7  557.85  5326.1  563.14  5331.5  564.41
  5354.6  565.03  5516.2  559.36  5567.9   560.7    5591  559.57  5710.4  562.07
#Mann= 7 ,-1 , 0
  3820.3      .1       0    4623     .05       0  4843.5      .1       0
  4921.4    .033       0  4928.6      .1       0  4997.6     .05       0
  5094.2      .1       0
Bank Sta=4329.78,5207.81
XS Rating Curve= 0 ,0
Exp/Cntr=0.3,0.1

Type RM Length L Ch R = 1 ,32698   ,46,46,46
BEGIN DESCRIPTION:
Mapping XS 2fb8af5e
END DESCRIPTION:
XS GIS Cut Line= 5
      1976629.89     13476873.44      1976994.49     13476313.51
      1977236.68     13476167.67      1977356.47     13475862.98
      1977588.18     13475279.81
#Sta/Elev= 30
  3872.8  560.49  3983.6  561.05  4164.8  552.93  4405.8551.6703  4522.8  550.33
  4523.5  549.53  4531.3  550.33 4558.06551.6698    4569  552.02  4584.5  555.71
  4590.3  553.97  4607.2  555.49  4621.4  555.57  4627.2  553.95  4658.3   555.1
  4664.1  553.61  4714.3  554.68  5046.4  552.71  5072.3  552.61  5078.9  553.96
  5103.3   552.6  5108.7  554.51  5133.1  552.13  5202.7  554.68  5211.4  552.91
  5295.1  561.51  5349.1  564.71  5579.3  559.18  5708.4  561.77  5778.6   566.1
#Mann= 7 ,-1 , 0
  3872.8      .1       0  4522.8     .07       0  4531.3      .1       0
  4607.2     .05       0  4714.3      .1       0  5046.4     .05       0
  5072.3      .1       0
Bank Sta=4405.8,4558.06
XS Rating Curve= 0 ,0
Exp/Cntr=0.3,0.1

Type RM Length L Ch R = 1 ,32652   ,205,205,205
BEGIN DESCRIPTION:
UNT 022 in RCW 61.0
END DESCRIPTION:
XS GIS Cut Line= 5
      1976626.44     13476899.43      1977023.14     13476331.73
      1977278.35     13476204.13      1977405.95     13475844.76
      1977609.09     13475290.04
#Sta/Elev= 30
  3831.2  560.78  3911.6  561.62  3983.1   560.7  4069.4  555.91  4155.8  552.89
    4521  549.98  4546.3   550.3  4551.9  552.23  4568.7  550.63  4574.3  551.73
  4593.1  550.78  4636.3  550.26 4812.79547.8854  4882.5  547.92  4989.4  545.55
  4990.1  544.75  4997.9  545.55  5019.2   547.1  5086.2  546.36 5130.37547.8856
  5222.1  552.06  5259.9  556.01  5376.6  562.84    5382  561.85  5401.8  562.34
  5437.7  560.36  5584.9   558.8  5604.8  560.05  5726.8  561.29  5781.2  565.06
#Mann= 5 ,-1 , 0
  3831.2      .1       0  4593.1     .05       0  4636.3      .1       0
  4989.4     .07       0  4997.9      .1       0
Bank Sta=4812.79,5130.37
XS Rating Curve= 0 ,0
Exp/Cntr=0.3,0.1

Type RM Length L Ch R = 1 ,32447   ,310,310,310
BEGIN DESCRIPTION:
Mapping XS 048b14ec
END DESCRIPTION:
XS GIS Cut Line= 3
      1977646.38     13477092.12      1977427.65     13476727.57
      1977660.15     13475301.33
#Sta/Elev= 30
  3948.5  568.52  4020.1  564.14    4057  559.83  4108.4   556.9  4136.7  556.59
  4237.8  551.79  4296.1  551.14  4318.3  549.36  4389.8  549.26  4416.8  548.03
  4446.2  548.63  4467.4  547.72 4702.23546.9575  4880.7   546.2  4923.4  547.31
  4997.2  545.02  5000.2  544.88  5000.9  544.08  5007.9  544.08  5008.7  544.88
  5065.2  546.25  5137.6  545.56 5180.24546.9583  5237.5  548.21  5255.5  550.25
  5378.5  554.21  5383.5  553.79  5409.7  555.19  5642.7  557.84  5818.7  563.09
#Mann= 5 ,-1 , 0
  3948.5      .1       0  4880.7     .07       0  4997.2      .1       0
  5000.2     .07       0  5008.7      .1       0
Bank Sta=4702.23,5180.24
XS Rating Curve= 0 ,0
Exp/Cntr=0.3,0.1

Type RM Length L Ch R = 1 ,32137   ,435,435,435
BEGIN DESCRIPTION:
UNT 022 in RCW 60.0
END DESCRIPTION:
XS GIS Cut Line= 3
        1978025.     13476974.98        1977825.       13476175.
      1977800.05     13475295.26
#Sta/Elev= 30
  4186.7     566  4238.2   563.4  4300.1  557.31  4333.6  556.04  4369.6  553.48
  4534.6  547.47  4615.8  546.28 4643.21545.8328  4701.6  544.89  4763.9  544.54
  4787.1  545.27  4915.5  545.25  4939.1  545.46  4988.1   544.4  5051.3  545.89
  5074.8  545.52  5151.4  544.92  5157.1   544.3  5157.9   543.5  5164.9   543.5
  5165.6   544.3  5201.4  545.76  5221.4  545.14 5306.89545.8328  5381.5  547.03
  5401.5  547.92  5491.5  548.63  5651.6  552.23  5811.6  559.32  5891.4  561.63
#Mann= 7 ,-1 , 0
  4186.7      .1       0  4615.8     .05       0  4701.6      .1       0
  4915.5     .07       0  5074.8      .1       0  5157.1     .07       0
  5165.6      .1       0
Bank Sta=4643.21,5306.89
XS Rating Curve= 0 ,0
Exp/Cntr=0.3,0.1

Type RM Length L Ch R = 1 ,31702   ,593,593,593
BEGIN DESCRIPTION:
UNT 022 in RCW 59.0
END DESCRIPTION:
XS GIS Cut Line= 3
      1978202.83     13476986.25        1978175.       13476425.
      1978188.94     13475482.74
#Sta/Elev= 30
  4417.6  568.57    4509  562.43    4529  560.34    4539  560.65  4619.1  555.83
  4639.1   554.1  4701.7  551.79  4876.5  544.76  4899.4  544.86 4936.25 543.634
  4999.5  542.96  5167.6  543.23  5279.6  542.86  5285.3  541.72    5286  540.92
  5293.1  540.92  5293.9  541.72 5308.59543.6341  5359.6  544.29  5459.6  548.71
  5519.6  552.31  5579.6  557.91  5609.6  559.56  5639.6  560.38  5699.6  559.46
  5719.6  559.98  5749.6  558.94  5789.6  558.51  5809.6  559.06  5921.9  558.99
#Mann= 5 ,-1 , 0
  4417.6      .1       0  4701.7     .05       0  5167.6      .1       0
  5285.3    .035       0  5293.9      .1       0
Bank Sta=4936.25,5308.59
XS Rating Curve= 0 ,0
Exp/Cntr=0.3,0.1

Type RM Length L Ch R = 1 ,31109   ,415,415,415
BEGIN DESCRIPTION:
UNT 022 in RCW 58.0
END DESCRIPTION:
XS GIS Cut Line= 3
      1978709.77     13477222.39       1978768.8     13476211.94
      1978341.96     13475559.54
#Sta/Elev= 30
  4210.8  563.26  4278.3  560.26  4438.6  556.63  4478.7  558.03  4518.7  557.12
  4588.8  560.77  4638.9  562.04    4679  559.51  4726.6  554.27  4731.6   554.6
  4749.1  553.12  4809.2  546.51  4877.6  543.86 4962.09 541.386  5009.6  540.47
  5179.8   540.9  5214.6  540.08  5215.4  539.28  5222.5  539.28  5223.3  540.08
  5295.4  541.12  5310.5  540.49 5443.22541.3859  5604.3  547.24  5721.2  552.74
  5744.8  552.71  5808.1   557.3  5823.2  556.87  5937.7  560.99  6002.6  561.87
#Mann= 5 ,-1 , 0
  4210.8      .1       0  4877.6     .05       0  5214.6    .035       0
  5223.3     .05       0  5604.3      .1       0
Bank Sta=4962.09,5443.22
XS Rating Curve= 0 ,0
Exp/Cntr=0.3,0.1

Type RM Length L Ch R = 1 ,30694   ,340,340,340
BEGIN DESCRIPTION:
UNT 022 in RCW 57.0
END DESCRIPTION:
XS GIS Cut Line= 3
      1979091.72     13477277.93      1979116.02     13475961.94
      1978335.95     13475188.81
#Sta/Elev= 30
    4045   561.7    4228  552.66    4328  549.79    4418  549.86    4458  553.42
    4488  554.42    4558  554.82    4608  554.11    4648  551.26    4678  546.16
    4728  542.81  4786.6  541.42 4877.12539.3888  5093.8  538.51  5094.6  537.71
  5101.7  537.71  5102.5  538.51 5423.34539.3887  5529.5  542.32  5593.1  541.25
  5748.7  541.41  5890.1  544.04  5911.3  545.95  5931.1  545.42    6173   552.2
  6250.7  553.07  6257.8  553.86  6307.3  554.79    6378   555.2  6459.5  557.33
#Mann= 5 ,-1 , 0
    4045      .1       0  4786.6     .05       0  5093.8     .03       0
  5102.5     .05       0  5931.1      .1       0
Bank Sta=4877.12,5423.34
XS Rating Curve= 0 ,0
Exp/Cntr=0.3,0.1

Type RM Length L Ch R = 1 ,30354   ,177,177,177
BEGIN DESCRIPTION:
Mapping XS 88f426ce
END DESCRIPTION:
XS GIS Cut Line= 4
      1979207.03     13476812.34      1979387.16     13476499.82
       1979391.5      13475898.7      1979226.88     13475248.87
#Sta/Elev= 30
    4374  547.02  4474.5  544.61  4560.8   541.1    4683  539.03  4698.2  538.98
  4749.5  538.33  4787.7  539.11  4849.5  538.79  4859.5  537.91 4900.86537.5342
  4995.1  535.91  4995.9  535.11  5003.1  535.11  5003.9  535.91  5126.2   536.7
  5249.5  538.61 5380.42537.5339    5521  538.14  5618.2  539.46  5732.5  543.75
  5803.9  545.75  5855.5  549.08  5886.4  549.68    5907  551.53  5912.1  550.91
  5927.7  552.29  5953.1  552.76    5989  556.48  5994.1  555.97  6006.2  558.07
#Mann= 8 ,-1 , 0
    4374      .1       0    4683     .05       0  4698.2      .1       0
  4787.7     .05       0  4995.1    .035       0  5003.9     .05       0
    5521      .1       0  5732.5     .05       0
Bank Sta=4900.86,5380.42
XS Rating Curve= 0 ,0
Exp/Cntr=0.3,0.1

Type RM Length L Ch R = 1 ,30177   ,153,153,153
BEGIN DESCRIPTION:
UNT 022 in RCW 56.0
END DESCRIPTION:
XS GIS Cut Line= 3
      1979133.38     13477257.09      1979591.72     13476375.14
      1979355.61     13475170.29
#Sta/Elev= 30
  3852.6   560.9  4114.2  549.02  4181.8  547.72  4256.2  544.22  4361.1  541.02
  4453.9  539.91  4534.4  539.71  4570.6  539.02 4967.05536.7401  5025.7  535.18
  5026.5  534.38  5033.7  534.38  5034.5  535.18    5183  537.01  5424.9  536.95
  5481.5  537.64    5509  535.97 5515.77536.7399  5605.2  538.79  5682.3  541.91
  5712.8  547.01  5738.9  549.32  5886.1  551.22  5916.6  553.29  5996.3   556.5
  6001.4  557.55  6028.7  558.94  6047.7  558.68  6052.8  559.93  6074.3  559.26
#Mann= 7 ,-1 , 0
  3852.6      .1       0  4453.9     .05       0  4534.4      .1       0
  4570.6     .05       0  5025.7     .03       0  5034.5     .05       0
  5605.2      .1       0
Bank Sta=4967.05,5515.77
XS Rating Curve= 0 ,0
Exp/Cntr=0.3,0.1

Type RM Length L Ch R = 1 ,30024   ,256,256,256
BEGIN DESCRIPTION:
Mapping XS 4d47a99d
END DESCRIPTION:
XS GIS Cut Line= 4
       1979406.7     13476844.87      1979697.49     13476367.45
      1979719.19     13475657.81      1979567.36     13475169.76
#Sta/Elev= 30
    4268  541.29    4303  541.49  4377.3  540.13  4388.7  540.16  4474.9  538.88
    4797  536.97  4849.5  535.93  4899.5  536.45 4947.48535.7406  5005.1  534.57
  5005.9  533.77  5013.1  533.77  5013.9  534.57  5149.6  536.03  5240.4  535.31
  5319.7  535.71  5349.7  535.08 5436.68535.7405  5509.8  537.14  5604.8   537.1
  5632.1  539.11  5637.6  538.77  5669.9  540.16  5686.5  539.18  5707.6  539.11
  5728.4   540.9  5812.2  543.47  5864.6  544.34  5902.9  546.48  6048.1  550.85
#Mann= 7 ,-1 , 0
    4268      .1       0  4377.3     .05       0  4388.7      .1       0
  4474.9     .05       0  5005.1     .03       0  5013.9     .05       0
  5637.6      .1       0
Bank Sta=4947.48,5436.68
XS Rating Curve= 0 ,0
Exp/Cntr=0.3,0.1

Type RM Length L Ch R = 1 ,29768   ,539,539,539
BEGIN DESCRIPTION:
UNT 022 in RCW 55.0
END DESCRIPTION:
XS GIS Cut Line= 3
      1979195.86     13477246.69      1980056.25     13476029.17
      1980424.96     13475825.02
#Sta/Elev= 30
  3699.4  560.58    3829  554.96  3921.9  548.89  4030.9  546.32  4057.9  543.72
  4087.5  542.32  4123.2  542.62  4219.9  540.66  4366.1  538.46  4371.4  538.42
 4892.33534.7498  4970.2  533.47  5106.8  534.33  5144.2  533.09    5145  532.29
  5152.2  532.29    5153  533.09  5209.6   533.6  5223.1  534.65    5235  533.88
 5253.94534.7498  5354.1  538.99  5370.2  538.31  5375.9  539.72  5383.1  538.96
  5391.9  540.45  5397.6  540.12  5478.9  545.53  5522.4  550.75  5611.7  554.59
#Mann= 7 ,-1 , 0
  3699.4      .1       0  4219.9     .05       0  4366.1      .1       0
  4371.4     .05       0  5144.2     .03       0    5153     .05       0
  5209.6      .1       0
Bank Sta=4892.33,5253.94
XS Rating Curve= 0 ,0
Exp/Cntr=0.3,0.1

Type RM Length L Ch R = 1 ,29229   ,640,640,640
BEGIN DESCRIPTION:
UNT 022 in RCW 54.0
END DESCRIPTION:
XS GIS Cut Line= 3
      1979400.71     13477136.45      1980376.44     13476448.92
      1980626.43     13475834.35
#Sta/Elev= 30
  3661.3  555.04  3708.3   554.3  3729.2  553.11  3764.9  546.45  3779.7   546.2
  3815.4  542.77  3930.6  540.07  4009.1  538.12  4109.8  537.05  4282.2  536.22
    4584  533.04  4662.8  532.86  4692.4  533.63 4829.96532.0204    4929  531.61
  4996.4  530.91  4997.3  530.11  5004.7  530.11  5005.5  530.91 5022.09532.0201
  5031.9  533.29  5049.1  533.33  5085.9  536.17  5204.3  541.95  5269.4  548.64
  5292.7  550.14  5340.8  551.47  5370.3  553.36  5423.8  553.76  5518.4  556.56
#Mann= 5 ,-1 , 0
  3661.3      .1       0  3930.6     .05       0    4929      .1       0
  4996.4     .07       0  5005.5      .1       0
Bank Sta=4829.96,5022.09
XS Rating Curve= 0 ,0
Exp/Cntr=0.3,0.1

Type RM Length L Ch R = 1 ,28589   ,209,209,209
BEGIN DESCRIPTION:
UNT 022 in RCW 53.0
END DESCRIPTION:
XS GIS Cut Line= 3
      1980996.23     13477327.44      1980996.23     13476473.23
      1980767.06     13475913.32
#Sta/Elev= 30
  4167.1  556.18  4359.5  553.83  4389.5  551.56  4399.5  550.01  4419.5  544.94
  4449.5  539.86  4459.5  540.75  4469.5  539.15  4489.5  538.55  4529.5  535.49
  4539.5  536.11  4559.5  535.62  4589.5  533.74  4619.4  534.09  4699.5  531.13
  4819.5  530.45 4894.03528.8403  5004.4  526.31  5005.3  525.51  5013.7  525.51
  5014.7  526.31  5036.7  527.41  5073.4  527.28 5131.78528.8405  5351.7  534.51
  5434.6  537.83    5464  539.82  5493.5  540.02    5512  540.09  5626.3  548.39
#Mann= 5 ,-1 , 0
  4167.1      .1       0  4619.4     .05       0  5004.4    .035       0
  5014.7     .05       0  5493.5      .1       0
Bank Sta=4894.03,5131.78
XS Rating Curve= 0 ,0
Exp/Cntr=0.3,0.1

Type RM Length L Ch R = 1 ,28380   ,562,562,562
BEGIN DESCRIPTION:
UNT 022 in RCW 52.0
END DESCRIPTION:
XS GIS Cut Line= 3
      1982058.71       13477274.      1981490.15     13477011.42
      1980778.35     13475707.17
#Sta/Elev= 30
  3764.8  553.03  3790.9  551.43  3820.2  546.54  3881.5  543.15  3889.1  542.23
  3894.6  543.21  3923.1  539.03  3968.9  537.23    4135  537.24  4165.4  533.07
  4330.6  529.41  4582.8  530.81  4827.7  529.69 4853.22528.4499  5013.3  526.09
  5014.2  525.29  5023.6  526.09 5148.85528.4497  5432.2  533.03  5594.3  537.96
  5639.1  539.68  5651.5   541.9  5697.1  545.16  5742.6   552.2  5748.3  549.99
  5764.4  549.75  5791.9  550.36  5813.8  552.77  5829.9  551.21  5876.9  552.57
#Mann= 5 ,-1 , 0
  3764.8      .1       0  3881.5     .05       0  5013.3    .035       0
  5023.6     .05       0  5594.3      .1       0
Bank Sta=4853.22,5148.85
XS Rating Curve= 0 ,0
Exp/Cntr=0.3,0.1

Type RM Length L Ch R = 1 ,27818   ,454,454,454
BEGIN DESCRIPTION:
UNT 022 in RCW 51.0
END DESCRIPTION:
XS GIS Cut Line= 3
      1982342.27     13477364.09        1981675.       13476275.
      1981226.78     13475554.14
#Sta/Elev= 30
  3733.9   545.6  3759.8  545.76  3775.2  541.46  3790.6  541.66  3796.5  544.87
  3803.2  545.94  3893.7   544.5    3986  544.24  4007.3  545.16  4080.8  544.52
  4102.1  545.17  4138.8  543.14  4160.1  543.28  4213.4  541.35  4291.6  538.29
  4471.7  533.68 4872.77526.7949    4976   525.8    5003  524.37  5003.9  523.57
  5012.6  523.57  5013.5  524.37  5055.4  526.41 5133.76526.7949  5213.6   528.4
  5460.4  528.57  5737.8   529.9  5780.3  530.86  5845.7   530.6    5860  530.67
#Mann= 6 ,-1 , 0
  3733.9     .05       0  3893.7      .1       0  4213.4     .05       0
    5003    .035       0  5013.5     .05       0  5845.7      .1       0
Bank Sta=4872.77,5133.76
XS Rating Curve= 0 ,0
Exp/Cntr=0.3,0.1

Type RM Length L Ch R = 1 ,27364   ,411,411,411
BEGIN DESCRIPTION:
UNT 022 in RCW 50.0
END DESCRIPTION:
XS GIS Cut Line= 3
      1982644.35     13477030.74        1982025.       13476025.
      1981509.46     13475350.88
#Sta/Elev= 30
    3830  533.42  3834.6  531.63  3848.5  532.12  3855.9  533.82  3871.3  532.35
  3892.5   531.9  3971.8  532.05  4118.5  529.52    4167   529.8  4329.1  528.68
  4371.7  529.14  4582.3  533.65  4698.2  534.14  4734.9  533.82  4792.9  531.88
  4808.3  530.66 4917.59525.4364  4939.6  524.32  4975.9  523.79  4992.3  522.64
  4993.2  521.84    5002  521.84  5002.8  522.64  5053.8  524.85  5103.6  524.51
  5250.1525.4362  5332.2  526.39  5525.3  526.89    5781   529.1  5859.8  530.43
#Mann= 3 ,-1 , 0
    3830     .05       0  4992.3    .035       0  5002.8     .05       0
Bank Sta=4917.59,5250.1
XS Rating Curve= 0 ,0
Exp/Cntr=0.3,0.1

Type RM Length L Ch R = 1 ,26953   ,452,452,452
BEGIN DESCRIPTION:
UNT 022 in RCW 49.0
END DESCRIPTION:
XS GIS Cut Line= 3
      1982917.78     13476798.97        1982375.       13475825.
      1981791.02     13475115.78
#Sta/Elev= 30
  3891.1  529.73  3896.2  529.73  3918.5  528.39  3925.9  528.36  3931.7  529.08
  3941.4  527.74  3953.4  526.98  4175.1  525.76 4264.32524.6475  4499.7  523.88
  4732.9  525.09  4873.5  524.47  4911.2   523.4  4960.4  523.01  4983.2  522.48
  4987.1  522.06  4987.9  521.26  4996.8  521.26  4997.7  522.06  5003.2  522.54
  5062.8  524.42  5097.9  523.71 5178.81524.6475  5567.1  526.63  5666.7   527.8
  5801.7  531.17  5894.2  534.84  5908.5  534.87  5922.1  536.45  5924.8  536.45
#Mann= 3 ,-1 , 0
  3891.1     .05       0  4987.1    .035       0  4997.7     .05       0
Bank Sta=4264.32,5178.81
XS Rating Curve= 0 ,0
Exp/Cntr=0.3,0.1

Type RM Length L Ch R = 1 ,26501   ,426,426,426
BEGIN DESCRIPTION:
UNT 022 in RCW 48.0
END DESCRIPTION:
XS GIS Cut Line= 3
      1983498.53     13476658.38        1982775.       13475675.
      1981904.78     13474930.06
#Sta/Elev= 30
  3793.5  537.71  4077.5  531.57  4098.3  532.56    4113  528.96  4127.6  529.51
  4133.8  531.01  4148.4  529.51  4213.2  528.06    4420  526.61  4534.9  523.77
 4623.24522.8354  4956.9  522.37  5001.8  521.43  5002.6  520.63  5011.5  520.63
  5012.4  521.43  5021.5  522.12 5120.06522.8353  5312.4  524.46  5468.3  524.51
  5511.1  525.79  5553.9  524.88  5738.3  527.13  5922.7   530.9  5986.4  533.65
  6070.9  535.59  6099.4  538.24    6128  538.68  6145.5  539.97  6159.9  540.13
#Mann= 4 ,-1 , 0
  3793.5     .05       0  5001.8    .035       0  5012.4     .05       0
  6145.5      .1       0
Bank Sta=4623.24,5120.06
XS Rating Curve= 0 ,0
Exp/Cntr=0.3,0.1

Type RM Length L Ch R = 1 ,26075   ,453,453,453
BEGIN DESCRIPTION:
UNT 022 in RCW 47.0
END DESCRIPTION:
XS GIS Cut Line= 3
      1984401.28     13476653.13        1983075.       13475425.
      1982175.61     13474693.95
#Sta/Elev= 30
  3248.7   545.2  3372.1  541.08  3499.6  534.79  3711.7   528.3  3959.5  526.72
  4065.5  528.24  4143.2  530.01  4164.7  531.35  4171.5  529.41  4185.7   529.1
  4193.1  529.38  4207.2  531.62  4228.2  530.93  4235.6  531.59  4292.3  528.76
  4299.1  526.98  4313.3  525.83 4497.74521.5255  4660.2  521.51  4801.4  520.14
  4921.6  521.16  5047.6  519.73  5048.4  518.93  5057.3  518.93  5058.2  519.73
 5172.42521.5253  5597.2  524.39  5702.7  525.89  6009.5  534.35  6215.3  542.59
#Mann= 3 ,-1 , 0
  3248.7     .05       0  5047.6    .035       0  5058.2     .05       0
Bank Sta=4497.74,5172.42
XS Rating Curve= 0 ,0
Exp/Cntr=0.3,0.1

Type RM Length L Ch R = 1 ,25622   ,434,434,434
BEGIN DESCRIPTION:
UNT 022 in RCW 46.0
END DESCRIPTION:
XS GIS Cut Line= 3
      1984526.27     13476381.41        1983375.       13475125.
      1982311.04     13474391.87
#Sta/Elev= 30
  3310.3  543.15  3330.1  541.97  3336.9  542.15  3358.4  540.66  3563.2   532.8
    3705  528.61  3839.4  526.62  3867.8  526.82  3875.1  526.24  4108.3  523.98
  4122.5  522.93    4144  522.67  4186.6  521.03  4387.3520.3723  4455.4   519.6
  4554.1   519.5    4675  520.13  4787.8  519.81  4830.3  520.62  4981.1  519.27
  4981.9  518.47  4990.8  518.47  4991.7  519.27 5127.49520.3724  5583.2  523.48
  5890.8  527.28  5949.5  528.69    6043  531.91  6135.6  533.29  6306.5  537.53
#Mann= 3 ,-1 , 0
  3310.3     .05       0  4981.1    .035       0  4991.7     .05       0
Bank Sta=4387.3,5127.49
XS Rating Curve= 0 ,0
Exp/Cntr=0.3,0.1

Type RM Length L Ch R = 1 ,25188   ,453,453,453
BEGIN DESCRIPTION:
UNT 022 in RCW 45.0
END DESCRIPTION:
XS GIS Cut Line= 3
      1984825.02     13475875.01        1983625.       13474775.
      1982530.66     13474166.17
#Sta/Elev= 30
  3354.5  547.23  3368.2  546.33  3396.8  545.43  3453.5  541.34  3475.1  538.89
  3517.3  537.68  3616.3  532.68  3963.4  524.15  3991.8  523.23  4005.7   521.6
  4026.9  521.71  4055.3  520.05 4087.23519.5506  4161.4  518.55  4339.8   518.1
  4340.6   517.3  4349.6   517.3  4350.4   518.1  4706.5  519.78  4755.8  518.71
  4869.3  519.58  4996.1  518.95 5093.32519.5505    5234   520.3  5607.9  524.67
  5732.6  527.13  5819.5  530.31  6084.8  536.24    6166  537.74  6234.7  537.59
#Mann= 4 ,-1 , 0
  3354.5      .1       0  3368.2     .05       0  4339.8    .035       0
  4350.4     .05       0
Bank Sta=4087.23,5093.32
XS Rating Curve= 0 ,0
Exp/Cntr=0.3,0.1

Type RM Length L Ch R = 1 ,24735   ,241,241,241
BEGIN DESCRIPTION:
UNT 022 in RCW 44.0
END DESCRIPTION:
XS GIS Cut Line= 3
      1985074.97     13475924.97        1983875.       13474425.
      1982630.47     13474001.23
#Sta/Elev= 30
  3051.3  564.62  3101.7  562.96  3136.9  558.56  3200.9  554.89  3323.3  542.75
  3378.6  538.68  3563.5  530.75  3783.6  524.99  3883.7   524.3  3905.3  522.18
  3934.1  522.63  3961.3  520.36 4011.57518.8467  4134.4  517.54  4135.3  516.74
  4145.1  517.54  4598.6  519.17  4671.5  518.98  4744.9  519.28  4937.2  518.89
  4993.3  518.36    5014  519.97 5031.19518.8469  5215.2   519.7  5484.3  524.61
  5578.4  527.78  5735.2  535.38    5892  539.96  6012.1  541.03  6286.9  536.16
#Mann= 8 ,-1 , 0
  3051.3      .1       0  3323.3     .05       0  4134.4    .035       0
  4145.1     .05       0  4598.6      .1       0  4671.5     .05       0
  4744.9      .1       0  4937.2     .05       0
Bank Sta=4011.57,5031.19
XS Rating Curve= 0 ,0
Exp/Cntr=0.3,0.1
