--- UNT 030 in RCW.prj (project) ---

Proj Title=UNT 030 in RCW Base Level Engineering
Current Plan=p01
Default Exp/Contr=0.3,0.1
English Units
Geom File=g01
Flow File=f01
Plan File=p01
Y Axis Title=Elevation
X Axis Title(PF)=Main Channel Distance
X Axis Title(XS)=Station
BEGIN DESCRIPTION:
UNT 030 in RCW
END DESCRIPTION:
DSS Export Rating Curves= 0
DSS Export Rating Curve Sorted= 0
DSS Export Volume Flow Curves= 0
DXF OffsetX= 0
DXF OffsetY= 0
DXF ScaleX= 1
DXF ScaleY= 10

--- UNT 030 in RCW.p01 (plan) ---

Plan Title=Multiple Run
Short Identifier=Multiple
Geom File=g01
Flow File=f01
Subcritical Flow
K Sum by GR= 0
Std Step Tol= 0.01
Critical Tol= 0.01
Num of Std Step Trials= 20
Max Error Tol= 0.3
Flow Tol Ratio= 0.001
Split Flow NTrial= 30
Split Flow Tol= 0.02
Split Flow Ratio= 0.02
Log Output Level= 0
Friction Slope Method= 1
Unsteady Friction Slope Method= 2
Unsteady Bridges Friction Slope Method= 1
Parabolic Critical Depth
Global Vel Dist=  1 , 1 , 1
Global Log Level= 0
CheckData=True
Encroach Param= -1, 0, 0, 0
BEGIN DESCRIPTION:
Multiple Run
END DESCRIPTION:

--- UNT 030 in RCW.f01 (steady flow) ---

Flow Title=Multiple
Program Version=5.05
Number of Profiles= 7
Profile Names=10-year,25-year,50-year,1pct_min,100-year,1pct_plu,500-year
River Rch & RM=UNT 030 in RCW,Reach-1         ,17890
     161     218     266     161     322     643     480
River Rch & RM=UNT 030 in RCW,Reach-1         ,17484
     258     359     444     273     545    1087     835
River Rch & RM=UNT 030 in RCW,Reach-1         ,11763
     310     432     533     328     654    1306    1001
River Rch & RM=UNT 030 in RCW,Reach-1         ,6086
     450     641     803     501     999    1993    1570
River Rch & RM=UNT 030 in RCW,Reach-1         ,3702
     450     641     803     501     999    1993    1570
River Rch & RM=UNT 030 in RCW,Reach-1         ,679
     450     641     803     501     999    1993    1570
Boundary for River Rch & Prof#=UNT 030 in RCW,Reach-1         , 1
Up Type= 0
Dn Type= 3
Dn Slope=0.005
Boundary for River Rch & Prof#=UNT 030 in RCW,Reach-1         , 2
Up Type= 0
Dn Type= 3
Dn Slope=0.005
Boundary for River Rch & Prof#=UNT 030 in RCW,Reach-1         , 3
Up Type= 0
Dn Type= 3
Dn Slope=0.005
Boundary for River Rch & Prof#=UNT 030 in RCW,Reach-1         , 4
Up Type= 0
Dn Type= 3
Dn Slope=0.005
Boundary for River Rch & Prof#=UNT 030 in RCW,Reach-1         , 5
Up Type= 0
Dn Type= 3
Dn Slope=0.005
Boundary for River Rch & Prof#=UNT 030 in RCW,Reach-1         , 6
Up Type= 0
Dn Type= 3
Dn Slope=0.005
Boundary for River Rch & Prof#=UNT 030 in RCW,Reach-1         , 7
Up Type= 0
Dn Type= 3
Dn Slope=0.005
DSS Import GetInterval= 0
DSS Import GetPeak= 0
DSS Import FillOption= 0

--- UNT 030 in RCW.g01 (geometry) ---

Geom Title=Existing Conditions
Program Version=5.05

River Reach=UNT 030 in RCW  ,Reach-1
Reach XY= 30
       2016400.8     13466904.54       2016720.8     13466723.92
      2016720.37      13466358.9       2016910.8     13466334.54
       2017000.8     13465294.54      2016822.45     13464903.61
      2016520.89     13464806.73      2016517.77     13464396.84
       2016310.8     13464284.54       2016110.8     13463604.54
       2015920.8     13463704.54       2015860.8     13463524.54
      2015193.29     13463390.07       2015300.8     13462914.54
       2014980.8     13462624.54      2015279.15     13461135.44
       2015707.4      13461163.2      2016297.68       13460250.
      2016142.12     13460009.03      2016199.43     13458594.49
       2016029.3     13458301.44       2015620.8     13458204.54
       2015270.8     13457584.54       2015490.8     13457254.54
       2015290.8     13456974.54       2015300.8     13456254.54
       2015480.8     13456094.54       2015300.8     13455694.54
       2015650.8     13455174.54       2015540.8     13454824.54

Type RM Length L Ch R = 1 ,17890   ,406,406,406
BEGIN DESCRIPTION:
UNT 030 in RCW 32.0
END DESCRIPTION:
XS GIS Cut Line= 3
      2016871.43     13467614.73      2016432.12     13466737.85
      2015983.23     13466288.96
#Sta/Elev= 30
  4120.1  488.23  4191.4  487.56  4230.5  485.36  4303.1  484.22  4309.9  483.54
  4459.5  482.82  4476.3  482.02  4610.4  480.65    4616  481.07  4655.1  480.06
  4677.4  480.32  4690.2  479.44  4779.7  478.69  4856.2  476.58  4891.5  474.52
  4923.3  473.78  4958.7  471.99  4990.3   471.8  4995.9  471.58  5000.4  470.39
  5000.9  469.59  5005.9  469.59  5006.4  470.39    5035  472.08  5079.7  473.04
  5221.1  473.31  5298.8  474.77  5468.5  478.58  5673.6  484.62  5735.7  485.13
#Mann= 3 ,-1 , 0
  4120.1      .1       0  5000.4     .07       0  5006.4      .1       0
Bank Sta=5000.4,5006.4
XS Rating Curve= 0 ,0
Exp/Cntr=0.3,0.1

Type RM Length L Ch R = 1 ,17484   ,647,647,647
BEGIN DESCRIPTION:
Mapping XS fb3bd62e
END DESCRIPTION:
XS GIS Cut Line= 2
      2017439.96     13467263.12      2016234.43       13466179.
#Sta/Elev= 30
  4031.5  487.48  4189.3  484.66  4260.3  481.88  4295.4  481.92  4302.9  481.07
  4309.6  481.31  4331.3  479.94  4380.6  479.68  4401.5   478.7  4472.6  478.13
    4480  477.63  4486.8     478  4614.6  474.54  4819.4  471.91  4947.2  471.55
  4982.3  471.12  4993.5  470.39    4994  469.59    4999  469.59  4999.5  470.39
  5018.2  470.83  5024.9  470.41  5145.3  470.44  5237.2  471.39  5329.3  473.66
  5385.9  476.72  5421.8  477.87  5463.7   480.4  5542.2  483.35  5652.8  486.12
#Mann= 3 ,-1 , 0
  4031.5      .1       0  4993.5     .07       0  4999.5      .1       0
Bank Sta=4993.5,4999.5
XS Rating Curve= 0 ,0
Exp/Cntr=0.3,0.1

Type RM Length L Ch R = 1 ,16837   ,483,483,483
BEGIN DESCRIPTION:
UNT 030 in RCW 31.0
END DESCRIPTION:
XS GIS Cut Line= 3
      2017625.01       13466475.        2016925.       13466325.
      2016425.02     13466125.01
#Sta/Elev= 30
  4268.8  490.15  4387.3  484.31  4392.4  484.56  4431.6  481.46  4436.7  481.99
  4442.7  480.63  4452.9  479.78    4481  478.35  4673.6  473.15  4818.5  471.47
  4923.3  470.26  4965.1  468.77  4974.5  468.13  4982.1  466.68  4996.4  466.41
  4996.9  465.61  5002.1  465.61  5002.6  466.41  5006.2  467.36    5017  468.02
  5092.4  467.85  5190.7  469.13  5209.5  469.59  5232.4  471.51  5239.2  470.87
  5286.3  472.08  5376.5  476.16  5437.1  480.16  5484.2  481.11  5523.2  483.66
#Mann= 4 ,-1 , 0
  4268.8     .05       0  4818.5      .1       0  4996.4     .07       0
  5002.6      .1       0
Bank Sta=4996.4,5002.6
XS Rating Curve= 0 ,0
Exp/Cntr=0.3,0.1

Type RM Length L Ch R = 1 ,16354   ,490,490,490
BEGIN DESCRIPTION:
UNT 030 in RCW 30.0
END DESCRIPTION:
XS GIS Cut Line= 3
      2018060.68      13465600.8        2017025.       13465875.
      2016425.03     13466024.99
#Sta/Elev= 30
  3913.9  494.34    3988  490.65  4002.5  490.52  4043.9  488.37  4068.4  487.82
  4143.7  484.01  4199.1  482.03  4271.5  477.92  4323.2  476.66  4339.7  475.85
  4570.7  470.87  4691.3  468.92  4731.6  468.83  4766.6  467.96  4861.1  467.12
  4992.4   464.7  4992.9   463.9  4998.2   463.9  4998.7   464.7  5132.2  466.99
  5250.7  471.49  5397.6  475.85  5420.8  476.83  5428.5   477.6  5490.3  478.89
  5523.4  480.21  5562.5  481.41  5572.8  481.29  5593.4  482.77  5603.7  482.97
#Mann= 4 ,-1 , 0
  3913.9     .05       0  4992.4     .03       0  4998.7     .05       0
  5523.4      .1       0
Bank Sta=4992.4,4998.7
XS Rating Curve= 0 ,0
Exp/Cntr=0.3,0.1

Type RM Length L Ch R = 1 ,15864   ,500,500,500
BEGIN DESCRIPTION:
UNT 030 in RCW 29.0
END DESCRIPTION:
XS GIS Cut Line= 3
      2017824.96     13465025.02        2017025.       13465425.
      2016274.96     13466025.03
#Sta/Elev= 30
  4112.1  494.77  4209.9  489.29  4327.3  484.13  4335.7  483.18  4388.8  480.04
  4433.5  474.72  4478.2  472.57  4612.4  468.82  4738.2  466.46  4858.3  464.92
  4953.4  464.46  4998.1  463.31  5034.5  464.14  5063.3  463.26  5103.4  463.11
  5103.9  462.31  5109.2  462.31  5109.7  463.11  5112.9  463.68  5148.2  464.08
  5276.2  468.43  5639.6  477.94  5674.8  479.97  5682.8  480.92  5689.2   480.3
  5716.7  480.41  5753.2  480.76  5761.3  481.71  5810.9  483.31    5967  487.38
#Mann= 4 ,-1 , 0
  4112.1     .05       0  5103.4     .03       0  5109.7     .05       0
  5716.7      .1       0
Bank Sta=5103.4,5109.7
XS Rating Curve= 0 ,0
Exp/Cntr=0.3,0.1

Type RM Length L Ch R = 1 ,15364   ,462,462,462
BEGIN DESCRIPTION:
UNT 030 in RCW 28.0
END DESCRIPTION:
XS GIS Cut Line= 3
      2017624.99     13464375.01        2016825.       13465025.
       2016151.6     13465760.66
#Sta/Elev= 30
  3978.6  494.05  4035.3  491.37  4176.8  486.07  4241.5   481.3  4305.4  478.44
  4348.5  475.04  4398.1  472.74  4426.8  472.31  4554.7  468.01  4674.6  464.66
  4789.6  462.58  4903.1     462  4955.9  461.02  4956.4  460.22  4961.8  460.22
  4962.3  461.02  4973.4  461.42  4995.7  461.14  5002.2   461.7  5065.8  461.12
  5101.6  461.47  5306.9  467.86  5327.9  467.98  5504.9  473.13  5582.6  473.71
  5639.3  475.09  5662.3  474.87  5809.2  477.99  5851.4  478.38  6006.7   482.6
#Mann= 4 ,-1 , 0
  3978.6     .05       0  4955.9     .03       0  4962.3     .05       0
  5662.3      .1       0
Bank Sta=4955.9,4962.3
XS Rating Curve= 0 ,0
Exp/Cntr=0.3,0.1

Type RM Length L Ch R = 1 ,14902   ,586,586,586
BEGIN DESCRIPTION:
UNT 030 in RCW 27.0
END DESCRIPTION:
XS GIS Cut Line= 3
      2017374.97     13464275.02        2016575.       13464825.
      2015909.74     13465559.68
#Sta/Elev= 30
  3996.7  486.76    4040  484.02  4105.6  481.33  4284.9  472.14  4457.8  466.34
  4529.8  463.25  4709.1  459.89  4873.4  460.66    4954  460.05  4992.3  458.61
  4992.8  457.81  4998.2  457.81  4998.7  458.61  5017.2  459.84  5137.5  462.69
  5165.9  463.14  5172.6   462.6  5186.8  463.67  5286.2  465.83  5321.3  465.64
  5349.7   466.5  5357.1  467.96  5378.1  469.22  5392.3  468.84  5406.5   469.8
  5413.2  468.57  5427.4   468.4  5503.2  470.32  5817.4  476.52  5958.6  480.75
#Mann= 4 ,-1 , 0
  3996.7     .05       0  4992.3     .03       0  4998.7     .05       0
  5503.2      .1       0
Bank Sta=4992.3,4998.7
XS Rating Curve= 0 ,0
Exp/Cntr=0.3,0.1

Type RM Length L Ch R = 1 ,14316   ,38,38,38
BEGIN DESCRIPTION:
Mapping XS 84f4f388
END DESCRIPTION:
XS GIS Cut Line= 6
        2016999.     13464032.26      2016681.31     13464402.03
      2016584.95     13464381.19      2016535.47      13464383.8
      2016418.29     13464435.88      2015759.74     13465365.14
#Sta/Elev= 30
  4340.3  475.59  4706.8  463.38  4911.3  458.99  4995.1  456.44  4997.1  455.76
  4997.6  454.96    5003  454.96  5003.5  455.76  5028.5  457.18  5033.8  458.84
  5037.4  456.78  5050.4  458.03  5056.2  456.54  5071.6  458.32  5135.9  457.39
  5142.1  458.38  5156.8  458.55  5192.5  457.66  5226.1  458.09  5394.3  460.32
  5658.9  467.45  5795.5  468.67    5825  469.89    5953  470.08  6003.4  471.15
  6011.2  472.17  6125.2  470.89    6140  472.14  6175.7  471.41  6244.3  472.27
#Mann= 6 ,-1 , 0
  4340.3     .05       0  4911.3      .1       0  4997.1     .07       0
  5003.5      .1       0  5226.1     .05       0  6011.2      .1       0
Bank Sta=4997.1,5003.5
XS Rating Curve= 0 ,0
Exp/Cntr=0.3,0.1

Type RM Length L Ch R = 1 ,14278   ,32,32,32
BEGIN DESCRIPTION:
UNT 030 in RCW 26.0
END DESCRIPTION:
XS GIS Cut Line= 6
      2016986.02     13463986.63      2016670.89     13464362.96
      2016522.45     13464344.73      2016459.56      13464376.2
      2016409.17      13464415.7      2015719.56     13465357.73
#Sta/Elev= 30
  4320.9  476.67  4761.1  461.61  4826.6  460.23    4869   461.4  4898.6  463.17
  4909.3  462.34  4948.8  463.02  4968.6  461.95  4980.9   462.7  4996.6  461.63
  5013.4  462.31  5018.9  461.41  5034.8  462.04    5049  461.31  5069.8  458.17
  5076.1  457.92  5141.7  458.51  5180.2  457.58  5180.7  456.78  5186.1  456.78
  5186.6  457.58  5221.7  458.09  5348.6  459.33  5670.5  467.93  6029.9   470.1
  6122.2  471.25  6178.5  470.43  6207.9  471.51  6228.7  471.19  6263.2  472.01
#Mann= 6 ,-1 , 0
  4320.9     .05       0    4869      .1       0  5180.2     .07       0
  5186.6      .1       0  5221.7     .05       0  6029.9      .1       0
Bank Sta=5180.2,5186.6
XS Rating Curve= 0 ,0
Exp/Cntr=0.3,0.1

Type RM Length L Ch R = 1 ,14246   ,415,415,415
BEGIN DESCRIPTION:
Mapping XS 809a7c96
END DESCRIPTION:
XS GIS Cut Line= 6
      2016957.38     13463982.72      2016652.66      13464326.5
      2016525.06      13464326.5      2016467.76     13464336.92
      2016407.87     13464362.96      2015666.65     13465351.25
#Sta/Elev= 30
  4353.7  475.65    4385  474.96  4413.5  472.49    4421  473.62  4441.9  471.21
  4449.4  472.47  4456.1  471.39  4505.5  471.47  4569.9  468.09  4838.2  460.69
  4920.7  459.63  4958.1  457.99  4963.2  458.85  4994.6  456.54  4995.1  455.74
    5001  456.54    5007  458.58  5030.5  458.18  5035.9  459.19  5075.2  456.92
  5110.6  458.11  5222.9  457.95  5339.8  458.97  5560.6  464.95  5589.8  466.09
    5596  467.36  5616.9  466.29  5666.9  467.77  6063.4  469.33  6299.6   470.7
#Mann= 6 ,-1 , 0
  4353.7     .05       0  4838.2      .1       0  4994.6     .07       0
    5001      .1       0  5222.9     .05       0  6063.4      .1       0
Bank Sta=4994.6,5001
XS Rating Curve= 0 ,0
Exp/Cntr=0.3,0.1

Type RM Length L Ch R = 1 ,13831   ,497,497,497
BEGIN DESCRIPTION:
UNT 030 in RCW 25.0
END DESCRIPTION:
XS GIS Cut Line= 3
      2016475.03     13463824.97        2016275.       13464075.
      2015074.99     13465175.01
#Sta/Elev= 30
  4674.1   473.6  4710.2  469.27    4731  465.99  4788.6   459.8  4879.8  456.15
  4943.9  455.21  4980.7  455.89  4991.1  454.54  4997.7  454.54  4998.2  453.21
  4998.7  452.41  5004.1  452.41  5004.6  453.21  5015.6   455.8    5171  455.21
  5262.7  456.41  5418.8  460.07  5539.1  461.32  5652.5  461.13    5766  461.87
  5801.2  460.47  5808.2  461.31  5836.3  462.14    5971   464.1  6183.8  469.63
  6204.4  470.25    6226  471.97  6261.2  472.01  6388.8  476.97  6622.2  483.04
#Mann= 5 ,-1 , 0
  4674.1      .1       0  4998.2     .07       0  5004.6      .1       0
  5262.7     .05       0  6183.8      .1       0
Bank Sta=4998.2,5004.6
XS Rating Curve= 0 ,0
Exp/Cntr=0.3,0.1

Type RM Length L Ch R = 1 ,13334   ,476,476,476
BEGIN DESCRIPTION:
UNT 030 in RCW 24.0
END DESCRIPTION:
XS GIS Cut Line= 3
      2016225.02     13463574.98        2016125.       13463675.
      2014893.51     13464743.85
#Sta/Elev= 30
  4855.9  470.97  4884.2  469.68  4898.4  468.24  4940.8  455.86  4983.2  451.76
  4990.6  450.43  4991.1  449.63  4996.6  449.63  4997.1  450.43  5000.7  450.43
  5004.5  452.52  5011.1  453.79  5103.3  454.13  5125.1  452.61  5188.7  454.21
  5337.8  453.95  5358.7  454.59  5550.5  455.12  5656.9  456.72  5904.7  458.46
  6060.5  461.39  6096.4  461.14  6138.3  463.01  6308.3  466.22  6322.5  465.71
  6344.4  466.86  6400.9  467.85  6428.9  469.44    6465   469.3    6628  476.36
#Mann= 3 ,-1 , 0
  4855.9      .1       0  4990.6     .07       0  4997.1      .1       0
Bank Sta=4990.6,4997.1
XS Rating Curve= 0 ,0
Exp/Cntr=0.3,0.1

Type RM Length L Ch R = 1 ,12858   ,522,522,522
BEGIN DESCRIPTION:
UNT 030 in RCW 23.0
END DESCRIPTION:
XS GIS Cut Line= 3
      2016169.59     13463413.09      2015243.37     13463937.83
      2014281.55     13464121.86
#Sta/Elev= 30
  4645.1  467.76  4700.9  467.54  4781.7   465.7  4811.3  463.49  4840.9  459.14
  4878.4  455.94  4937.5   452.3  4972.2  451.39  4980.8  449.11  4986.6  450.99
  4991.9  448.28  4992.4  447.48  4997.9  447.48  4998.4  448.28  5002.5  452.52
  5024.1  453.22  5098.6  452.27  5384.8  452.33  5661.8  454.27  5883.5  452.57
    6156  454.73  6310.1  459.42  6357.1  462.34  6362.2   461.8  6409.2  465.59
  6414.3  464.72  6461.2  467.61  6466.3  467.14  6518.4  469.61  6688.9  474.18
#Mann= 3 ,-1 , 0
  4645.1      .1       0  4991.9     .07       0  4998.4      .1       0
Bank Sta=4991.9,4998.4
XS Rating Curve= 0 ,0
Exp/Cntr=0.3,0.1

Type RM Length L Ch R = 1 ,12336   ,573,573,573
BEGIN DESCRIPTION:
UNT 030 in RCW 22.0
END DESCRIPTION:
XS GIS Cut Line= 3
      2016005.94     13463158.77       2015239.9      13463649.2
      2014625.03       13463675.
#Sta/Elev= 30
  4378.6  468.25  4471.2  463.38  4534.6  457.87  4593.4  454.85  4664.9   453.3
  4783.2  451.92  4934.6  451.99  4970.9  451.46  4985.3  450.99  4992.1  449.53
  4994.8  446.92  4995.3  446.12  5000.8  446.12  5001.3  446.92  5013.2  450.74
  5028.4  450.55  5034.4  451.16  5049.6  450.16  5056.5  450.95  5122.3  450.32
  5333.1  451.68  5533.3  451.94  5573.3  450.83  5583.3  449.26  5653.4  454.57
  5713.5  457.43  5781.4   465.1  5813.5  467.08  5883.6  473.25  5903.6  476.21
#Mann= 3 ,-1 , 0
  4378.6      .1       0  4994.8     .07       0  5001.3      .1       0
Bank Sta=4994.8,5001.3
XS Rating Curve= 0 ,0
Exp/Cntr=0.3,0.1

Type RM Length L Ch R = 1 ,11763   ,21,21,21
BEGIN DESCRIPTION:
Mapping XS 349aa6e5
END DESCRIPTION:
XS GIS Cut Line= 6
      2015937.83     13463152.67       2015343.2     13463261.18
      2015226.01     13463239.48      2015150.06     13463211.27
      2015100.14     13463224.29       2014260.3     13463200.42
#Sta/Elev= 30
  4199.3  465.73  4334.3  459.75  4385.1  455.38  4415.6  453.76  4573.8  450.93
  4649.4  450.83  4679.9  450.06  4863.3  449.97  4893.9  450.69  4913.2  450.27
  4918.2     451  4935.4  449.78  4942.6   448.5  4948.2  449.88  4957.7  448.65
    4979  449.63  5006.2  448.21  5006.8  447.41    5013  447.41  5013.5  448.21
  5081.4  449.81  5111.4  449.29  5151.4  451.13  5221.4  451.83  5331.5  454.47
  5557.9  462.79  5591.6   463.3  5671.6     467  5851.7   468.6  5896.4  470.44
#Mann= 3 ,-1 , 0
  4199.3      .1       0  5006.2     .07       0  5013.5      .1       0
Bank Sta=5006.2,5013.5
XS Rating Curve= 0 ,0
Exp/Cntr=0.3,0.1

Type RM Length L Ch R = 1 ,11742   ,34,34,34
BEGIN DESCRIPTION:
Mapping XS 2c3eabd4
END DESCRIPTION:
XS GIS Cut Line= 6
      2016002.89     13463126.64      2015358.39     13463241.65
      2015254.22     13463226.46      2015202.14     13463200.42
      2015124.01     13463185.23      2014249.72     13463163.54
#Sta/Elev= 30
  4137.5  468.77    4308  461.79  4419.8  454.43  4502.1  452.27  4683.9  450.01
    4836  449.73  4866.3  449.87  4886.6  451.95    4935  453.11  4955.7  452.48
  4957.9  451.53    4963  452.91  5003.7  451.96  5024.1  452.85  5076.7  451.77
  5100.9  449.04  5101.4  448.24  5107.6  448.24  5108.2  449.04  5144.5  452.08
  5174.6  451.22  5214.6   451.4  5304.6  453.42  5604.8  462.63  5654.8  464.89
  5724.8  464.81  5744.8  465.99  5774.9  465.04  5864.9  467.51  5910.2  469.66
#Mann= 3 ,-1 , 0
  4137.5      .1       0  5100.9     .07       0  5108.2      .1       0
Bank Sta=5100.9,5108.2
XS Rating Curve= 0 ,0
Exp/Cntr=0.3,0.1

Type RM Length L Ch R = 1 ,11708   ,499,499,499
BEGIN DESCRIPTION:
UNT 030 in RCW 21.0
END DESCRIPTION:
XS GIS Cut Line= 6
      2016175.04     13463074.99      2015410.47     13463219.95
       2015302.4     13463205.63      2015190.42     13463157.45
      2015029.83     13463160.92      2014119.14      13463128.4
#Sta/Elev= 30
  3965.9  472.82  4128.8  469.15  4240.7  465.02  4362.9  459.35  4425.6  454.58
    4485  452.97  4687.1  449.99  4948.5  449.69  4966.6  450.52  4971.8  448.92
  4980.4  449.09  4990.4  446.31  4996.8  445.82  4997.3  445.02  5003.5  445.02
  5004.1  445.82  5010.4  448.35  5050.4  447.21  5089.2  448.67  5100.5  448.22
  5135.5  451.17  5210.5  451.04  5310.6  453.17  5550.7  460.63  5730.8  464.37
  5760.9  466.33  5790.9  463.91  5810.9  466.23    5941  469.65  6046.9  474.96
#Mann= 3 ,-1 , 0
  3965.9      .1       0  4996.8     .07       0  5004.1      .1       0
Bank Sta=4996.8,5004.1
XS Rating Curve= 0 ,0
Exp/Cntr=0.3,0.1

Type RM Length L Ch R = 1 ,11209   ,460,460,460
BEGIN DESCRIPTION:
UNT 030 in RCW 20.0
END DESCRIPTION:
XS GIS Cut Line= 3
      2016091.03     13462822.38      2015329.31     13462759.45
      2014150.88     13462943.92
#Sta/Elev= 30
  4092.5  467.49  4128.7  465.76  4198.9   465.2  4399.6  459.17  4469.8  457.92
  4660.5   450.7    4811   446.6    4831  447.62  4899.1     448  4942.2  448.28
  4962.4  447.38  4972.5  448.04  4982.6  447.46  4988.7  445.06  4990.1  442.89
  4990.7  442.09  4996.9  442.09  4997.4  442.89  4999.1  443.83  5002.6  445.76
  5023.1   447.3  5195.2  446.77  5215.4  448.25  5286.3  448.27  5357.1  450.01
  5407.8  452.61  5442.8   452.8  5630.4  461.13  5964.6  472.46  6049.6  477.15
#Mann= 6 ,-1 , 0
  4092.5      .1       0  4899.1     .07       0  4990.1     .07       0
  4997.4     .07       0  4999.1     .07       0  5002.6      .1       0
Bank Sta=4990.1,4997.4
XS Rating Curve= 0 ,0
Exp/Cntr=0.3,0.1

Type RM Length L Ch R = 1 ,10749   ,560,560,560
BEGIN DESCRIPTION:
UNT 030 in RCW 19.0
END DESCRIPTION:
XS GIS Cut Line= 3
      2016045.47     13462711.71        2015075.       13462525.
      2014475.05     13462425.01
#Sta/Elev= 30
    4038  463.27  4050.4   462.5  4211.6  459.68  4263.2  457.85    4310   457.6
  4323.6  456.36  4374.5  455.59  4445.8  452.62  4470.9  452.49  4588.4  448.82
  4700.4  447.31  4822.6  446.81  4863.3  445.47  4873.5   446.3    4903  446.62
  4975.4  446.99  4996.6  441.87  4997.2  441.07  5003.4  441.07    5004  441.87
  5005.9  444.53  5023.7  446.46  5101.8  446.42  5158.1  446.97  5279.7  450.15
  5302.5  451.39  5381.1  458.39  5452.1  460.43  5573.7   467.8  5634.5   474.3
#Mann= 5 ,-1 , 0
    4038      .1       0    4903     .12       0  4996.6     .07       0
    5004     .12       0  5101.8      .1       0
Bank Sta=4996.6,5004
XS Rating Curve= 0 ,0
Exp/Cntr=0.3,0.1

Type RM Length L Ch R = 1 ,10189   ,394,394,394
BEGIN DESCRIPTION:
UNT 030 in RCW 18.0
END DESCRIPTION:
XS GIS Cut Line= 3
      2016012.86     13462334.09        2015125.       13462175.
      2014441.72     13461997.73
#Sta/Elev= 30
  4130.5  462.63  4189.3  457.63  4341.7  451.97  4412.8  450.89  4514.4  448.06
  4585.5   447.6  4609.1  446.73  4900.4  444.51  4971.5  445.25  4981.7  444.74
  4988.2  441.42  4988.7  440.62    4995  440.62  4995.6  441.42  5000.6  442.12
  5005.6  441.55  5012.2  443.82  5022.3  444.73  5053.3  445.11  5104.8  444.95
    5164   445.9  5253.1  447.14  5404.4  451.66  5450.8  454.23  5466.4  452.89
  5476.7  452.93  5507.7  455.11  5572.5   457.3    5689  463.78  5738.4  465.62
#Mann= 5 ,-1 , 0
  4130.5      .1       0  4988.2     .07       0  4995.6      .1       0
  5053.3     .07       0    5164      .1       0
Bank Sta=4988.2,4995.6
XS Rating Curve= 0 ,0
Exp/Cntr=0.3,0.1

Type RM Length L Ch R = 1 ,9795    ,370,370,370
BEGIN DESCRIPTION:
UNT 030 in RCW 17.0
END DESCRIPTION:
XS GIS Cut Line= 3
      2015925.01     13462275.01      2015433.48      13461956.5
        2014420.     13461680.88
#Sta/Elev= 30
  4048.8  456.39  4077.5  455.86  4128.9  453.08    4274  448.16  4403.9  445.51
 4533.18444.2679  4746.9  443.65  4954.2  444.69  4974.9  444.03  4985.3  442.48
  4991.9  439.47  4992.5  438.67  4998.8  438.67  4999.3  439.47  5001.5  441.12
  5006.7  439.88  5016.4  441.29  5026.7  443.92 5060.05444.2676  5088.9  444.89
  5109.6  446.13  5115.7  447.24  5120.9  447.29  5150.3  450.83  5171.8  454.03
  5195.2  456.38  5213.3  457.47  5418.4  462.45  5577.5  464.11  5684.8  466.59
#Mann= 3 ,-1 , 0
  4048.8      .1       0  4991.9     .07       0  4999.3      .1       0
Bank Sta=4533.18,5060.05
XS Rating Curve= 0 ,0
Exp/Cntr=0.3,0.1

Type RM Length L Ch R = 1 ,9425    ,387,387,387
BEGIN DESCRIPTION:
UNT 030 in RCW 16.0
END DESCRIPTION:
XS GIS Cut Line= 3
      2016075.82     13462184.35      2015466.03     13461696.08
      2014432.15     13461589.87
#Sta/Elev= 30
    4006  461.16    4034  458.86  4162.1  453.03  4205.3  452.37  4290.1  448.86
  4432.6  445.23 4578.86443.1101  4760.7  442.05  4868.6  442.64  4918.9  441.95
  4949.3  443.47  4969.2  443.41  4979.2  441.85  4989.3  438.52  4995.6   437.5
  4996.2   436.7  5002.5   436.7    5003   437.5 5009.67443.1097  5019.4  443.82
  5079.7   444.2  5170.2  443.75  5270.7  445.78    5331  449.46    5336  449.22
  5430.2  457.02    5502   459.9  5733.2  461.82  5821.9  464.18  5826.5  463.71
#Mann= 3 ,-1 , 0
    4006      .1       0  4995.6     .07       0    5003      .1       0
Bank Sta=4578.86,5009.67
XS Rating Curve= 0 ,0
Exp/Cntr=0.3,0.1

Type RM Length L Ch R = 1 ,9038    ,411,411,411
BEGIN DESCRIPTION:
Mapping XS 363df18d
END DESCRIPTION:
XS GIS Cut Line= 4
      2016104.01     13462099.69      2015698.23     13461711.27
       2014988.6     13461218.65      2014630.84     13460949.79
#Sta/Elev= 30
    3838  458.32  3975.1  452.99  3982.1  452.15  4222.7  445.71 4436.08 442.634
  4671.5  440.13  4694.9  441.22  4715.8  440.32  4751.6  441.79  4793.5  442.25
  4951.6  442.75  4975.2  442.04  4981.3  442.74  4992.4  437.29    4993  436.49
  4999.3  436.49  4999.8  437.29    5011  440.38  5046.8  442.85  5103.5  442.03
 5212.92442.6343  5231.8  442.96  5276.2  445.57  5282.4  446.59  5311.6   447.6
  5440.7     455  5511.5  460.06  5576.1  460.76  5668.4  458.68  5711.1   458.8
#Mann= 3 ,-1 , 0
    3838      .1       0  4992.4     .07       0  4999.8      .1       0
Bank Sta=4436.08,5212.92
XS Rating Curve= 0 ,0
Exp/Cntr=0.3,0.1

Type RM Length L Ch R = 1 ,8627    ,372,372,372
BEGIN DESCRIPTION:
Mapping XS 275b96fc
END DESCRIPTION:
XS GIS Cut Line= 4
       2016095.4       13462039.      2015698.23     13461518.13
      2015298.93     13461053.72      2014671.78     13460812.84
#Sta/Elev= 30
  3873.9  455.56  4127.2  448.02 4387.63442.6047    4520  439.59  4561.4  439.06
  4583.4  439.81    4647  437.54  4774.3  440.24  4980.6  441.75  4987.2  436.46
  4997.8  435.21  4998.3  434.41  5004.6  434.41  5005.2  435.21    5008  437.98
    5030  441.94  5050.8  440.86  5100.2  442.18  5211.4  441.09    5242  441.94
  5290.7  439.11 5387.23442.6047  5430.1  446.12  5460.1  446.52  5484.7  449.75
  5531.2  452.55  5624.1  455.41  5678.8  455.42  5714.1  453.96  5813.2  457.79
#Mann= 3 ,-1 , 0
  3873.9      .1       0  4997.8     .07       0  5005.2      .1       0
Bank Sta=4387.63,5387.23
XS Rating Curve= 0 ,0
Exp/Cntr=0.3,0.1

Type RM Length L Ch R = 1 ,8255    ,35,35,35
BEGIN DESCRIPTION:
Mapping XS 48e20beb
END DESCRIPTION:
XS GIS Cut Line= 6
      2016140.92     13461975.99      2015745.98      13461207.8
       2015700.4     13461140.52      2015617.94     13461129.67
      2015392.24     13460977.76      2014748.86     13460516.34
#Sta/Elev= 30
  4072.1  455.94  4187.4  451.63 4609.56442.6012  4924.6   438.9  4952.3  434.16
  5000.3  433.34  5000.9  432.54  5007.8  433.34  5024.9  435.05  5053.3  433.81
  5093.5  435.89  5100.8  439.81  5105.6  439.81  5114.2  435.87  5120.3  437.08
  5128.5  435.71  5135.3  437.26  5141.3  435.59  5171.2  437.42  5177.3  440.08
  5243.2  440.73  5422.7  441.36  5523.4  439.54  5544.3  437.37  5594.6   440.1
  5624.1  439.07 5728.13442.6011  5888.1  446.16  6053.9   453.1  6164.6  455.65
#Mann= 3 ,-1 , 0
  4072.1      .1       0  5000.3     .07       0  5007.8      .1       0
Bank Sta=4609.56,5728.13
XS Rating Curve= 0 ,0
Exp/Cntr=0.3,0.1

Type RM Length L Ch R = 1 ,8220    ,38,38,38
BEGIN DESCRIPTION:
UNT 030 in RCW 15.0
END DESCRIPTION:
XS GIS Cut Line= 6
      2016175.01     13461975.02      2015763.77     13461158.32
      2015709.08     13461104.93      2015632.26      13461086.7
      2015380.96      13460956.5      2014840.19     13460474.75
#Sta/Elev= 30
  4033.9  457.08  4078.7  454.27    4338  447.88  4739.8  440.03  4861.6  439.03
  4892.6  441.98  4951.3  442.39  4971.4  440.86  4978.4  442.24  4985.5  441.16
  4992.5  442.43    5104  442.92  5123.9  439.02  5201.1  440.22  5228.9  438.09
  5245.4  440.29  5406.8  441.53    5477  438.69  5484.6  439.51  5509.2     437
  5509.8   436.2  5516.7     437  5519.7  438.77  5541.4  440.48    5605  439.73
  5611.7  438.44  5625.9  440.44  5668.5  440.26  5796.4  444.72  6111.3   452.1
#Mann= 3 ,-1 , 0
  4033.9      .1       0  5509.2     .07       0  5516.7      .1       0
Bank Sta=5509.2,5516.7
XS Rating Curve= 0 ,0
Exp/Cntr=0.3,0.1

Type RM Length L Ch R = 1 ,8182    ,293,293,293
BEGIN DESCRIPTION:
Mapping XS 19368901
END DESCRIPTION:
XS GIS Cut Line= 6
      2016198.24     13461966.05      2015830.18     13461198.68
      2015760.73     13461097.99      2015698.23     13461059.79
      2015628.79     13461063.27      2014854.49     13460441.74
#Sta/Elev= 30
  4006.4  457.16    4053  454.59  4585.1  442.13  4750.6  439.38  4950.6  437.69
  4978.9  436.73  4983.1  434.87  4983.7  434.07    4990  434.07  4990.6  434.87
  5009.6  437.29  5139.2  439.13    5160  438.43  5166.4  436.66  5209.7  435.73
  5230.5  436.64    5253  439.95  5302.6  440.51  5395.5  439.72  5416.3  436.52
  5445.2  439.71  5530.1  440.84  5600.6  438.32    5772  443.64  5786.4   445.6
  5807.2  442.47  5821.6  442.43    5843  445.23  5885.7  447.67  6116.1  452.78
#Mann= 3 ,-1 , 0
  4006.4      .1       0  4983.1     .07       0  4990.6      .1       0
Bank Sta=4983.1,4990.6
XS Rating Curve= 0 ,0
Exp/Cntr=0.3,0.1

Type RM Length L Ch R = 1 ,7889    ,711,711,711
BEGIN DESCRIPTION:
UNT 030 in RCW 14.0
END DESCRIPTION:
XS GIS Cut Line= 3
      2016270.29     13461494.73      2016141.38      13461003.8
      2015175.02     13460425.01
#Sta/Elev= 30
  4236.5  453.54  4284.7  453.11  4360.6   451.9  4525.7  443.99  4742.7  439.41
  4886.6  437.05  4914.7  435.52  4987.7  435.83  4996.3  434.27  4999.6  432.16
  5000.1  431.36  5007.1  432.16  5009.1  435.71  5067.5  436.85  5089.5  436.95
  5112.9  433.94  5139.7  433.82  5255.5  434.08  5322.7  438.42  5462.6   438.1
  5475.8  435.44  5485.5  434.87  5497.5  436.15  5512.7   435.1  5549.7  436.97
  5592.5  436.38  5650.8     443  5703.3  446.34  5746.1  452.48  5870.5  457.89
#Mann= 7 ,-1 , 0
  4236.5      .1       0  4284.7     .05       0  4742.7      .1       0
  4999.6     .07       0  5007.1      .1       0  5139.7     .05       0
  5255.5      .1       0
Bank Sta=4999.6,5007.1
XS Rating Curve= 0 ,0
Exp/Cntr=0.3,0.1

Type RM Length L Ch R = 1 ,7178    ,518,518,518
BEGIN DESCRIPTION:
UNT 030 in RCW 13.0
END DESCRIPTION:
XS GIS Cut Line= 3
        2016275.       13461375.       2016498.8     13460416.57
      2015353.47      13459929.8
#Sta/Elev= 30
  3771.9   452.7  3923.3  446.88  4160.5   442.7  4368.9  439.29  4412.8  438.64
    4822  436.92  4922.1  435.47  4966.7  432.92  4980.2  433.66  4988.4  433.18
  4994.6  430.41  4995.2  429.61  5002.2  430.41  5010.2  434.27    5021  434.84
  5135.8  434.38  5180.3  432.78  5227.5  434.11  5262.1  431.66  5309.4  431.15
  5314.8  432.51    5333  432.05    5344  433.68  5385.8  435.17  5651.2  436.32
  5683.8  437.28  5714.9   442.3  5738.2  444.26  5867.7  445.05  6000.6  451.62
#Mann= 8 ,-1 , 0
  3771.9     .05       0  4160.5      .1       0  4368.9     .05       0
  4412.8      .1       0  4994.6     .07       0  5002.2      .1       0
  5135.8     .05       0    5344      .1       0
Bank Sta=4994.6,5002.2
XS Rating Curve= 0 ,0
Exp/Cntr=0.3,0.1

Type RM Length L Ch R = 1 ,6660    ,574,574,574
BEGIN DESCRIPTION:
UNT 030 in RCW 12.0
END DESCRIPTION:
XS GIS Cut Line= 4
      2016420.92     13461450.16      2016561.54      13460267.9
       2016248.8      13459874.9      2015425.05       13459875.
#Sta/Elev= 30
  3244.6  451.75  3323.2  450.19  3368.3  449.06  3582.1  443.99    3844  439.62
  4015.2   438.2  4257.3  437.92  4594.7  435.72    4784  434.16  4861.1  432.62
  4961.2  433.34  4987.4  429.65    4988  428.85  4994.5  428.85  4995.1  429.65
  5011.2  431.47  5031.2  430.61  5061.2  431.81  5071.2  430.78  5101.2  430.86
  5121.2  431.99  5141.2  431.46  5201.2  433.73  5377.6  434.83  5461.2  435.84
  5511.2  442.94  5551.2  444.11  5601.2  444.24  5651.2  448.33  5761.2  451.23
#Mann= 7 ,-1 , 0
  3244.6      .1       0  3323.2     .05       0  3368.3      .1       0
  4594.7     .05       0  4987.4    .035       0  4995.1     .05       0
  5377.6      .1       0
Bank Sta=4987.4,4995.1
XS Rating Curve= 0 ,0
Exp/Cntr=0.3,0.1

Type RM Length L Ch R = 1 ,6086    ,63,63,63
BEGIN DESCRIPTION:
UNT 030 in RCW 11.0
END DESCRIPTION:
XS GIS Cut Line= 6
      2017326.92     13459830.63      2016990.98     13459726.46
      2016767.03     13459419.17      2016532.65     13459270.73
      2016319.11     13459268.13      2015388.38     13459652.86
#Sta/Elev= 30
  3651.1  463.06  3954.3  446.59  4221.3  436.53    4310   435.6  4381.4  434.46
  4401.7   434.9  4432.2  430.65  4438.2  432.62  4449.6  428.68  4450.2  427.88
  4457.3  428.68  4459.3  430.98  4463.6  430.43  4474.6   429.1  4495.8  431.78
    4511  429.35  4568.7  432.64  4610.1  431.22  4657.5  432.13  4738.4  430.94
  4813.6  430.71  4873.6  433.48  4881.8  431.37  4907.8  433.03  4944.4  430.82
  5124.7  432.61  5329.8  434.16  5504.5  441.38  5574.7  446.87  5881.8  452.08
#Mann= 12 ,-1 , 0
  3651.1      .1       0  4221.3     .16       0    4310      .1       0
  4381.4     .16       0  4449.6    .035       0  4457.3     .16       0
  4463.6     .05       0  4610.1     .16       0  4657.5     .05       0
  4738.4      .1       0  4813.6     .05       0  5124.7      .1       0
Bank Sta=4449.6,4457.3
XS Rating Curve= 0 ,0
Exp/Cntr=0.3,0.1

Type RM Length L Ch R = 1 ,6023    ,61,61,61
BEGIN DESCRIPTION:
Mapping XS b2717543
END DESCRIPTION:
XS GIS Cut Line= 6
      2017355.63     13459820.56      2017038.83     13459651.31
      2016769.73     13459356.17      2016448.55     13459182.56
      2016140.39     13459260.68      2015385.81     13459590.27
#Sta/Elev= 30
  3612.2  465.83  3720.1  461.94  4063.3  441.51  4098.9  441.23  4148.2  445.86
  4370.4  443.96  4417.8     444  4432.6  441.53  4453.6  443.37  4468.4  441.04
  4510.1   442.8  4576.7  444.55  4601.1  442.73  4770.3  444.59    4867  441.79
  4936.9  443.75  4942.1  441.58  4976.5  444.13  5118.1  444.51  5329.9  442.95
  5376.8  444.81  5382.2     443  5400.2  444.78    5454  440.95  5454.6  440.15
  5461.7  440.95  5533.5  441.86  5574.9  446.62  5650.6  449.29  5880.2  451.16
#Mann= 7 ,-1 , 0
  3612.2      .1       0  4370.4     .05       0  4510.1      .1       0
  4601.1     .05       0  5118.1      .1       0    5454     .03       0
  5461.7      .1       0
Bank Sta=5454,5461.7
XS Rating Curve= 0 ,0
Exp/Cntr=0.3,0.1

Type RM Length L Ch R = 1 ,5962    ,331,331,331
BEGIN DESCRIPTION:
UNT 030 in RCW 10.0
END DESCRIPTION:
XS GIS Cut Line= 6
      2017300.89     13459729.07      2016964.94     13459507.71
      2016780.05     13459275.94      2016600.36     13459153.54
      2016368.59     13459114.48      2015318.27     13459564.18
#Sta/Elev= 30
  3657.5  466.62  3765.6  459.68  3816.8  453.55  3988.4  445.88  4033.6  441.35
  4097.5   443.4    4140  437.33  4211.2  435.15  4367.7  431.97  4418.5  434.32
  4439.5  432.73  4454.4  435.46  4475.4  433.33  4490.3  435.63  4564.1  430.96
  4564.7  430.16  4571.8  430.96  4650.1  434.66  4731.3  434.01  4820.9  431.43
  4880.6  434.37  5043.4  434.42  5097.7  432.05  5322.2  434.49  5381.8  442.09
  5421.8  439.23  5535.8  441.61    5580  447.12  5646.3   448.9  5951.9  451.08
#Mann= 5 ,-1 , 0
  3657.5      .1       0  4564.1     .03       0  4571.8      .1       0
  4731.3     .05       0  5322.2      .1       0
Bank Sta=4564.1,4571.8
XS Rating Curve= 0 ,0
Exp/Cntr=0.3,0.1

Type RM Length L Ch R = 1 ,5631    ,419,419,419
BEGIN DESCRIPTION:
UNT 030 in RCW 9.0
END DESCRIPTION:
XS GIS Cut Line= 3
      2017861.37     13458775.72      2016477.96     13458744.69
      2015388.43     13459181.54
#Sta/Elev= 30
  3318.6  451.61  3905.1  436.98  4045.1  431.65  4065.2  428.36  4075.2  428.55
  4095.2  431.88  4105.2  432.21  4135.2  429.68  4285.2  427.72  4365.2  429.48
  4385.2  428.46  4395.2  426.86  4415.2   429.4  4435.2  429.33  4455.3  428.55
  4471.4  424.45    4472  423.65  4478.5  423.65  4479.2  424.45  4495.3  428.66
  4515.3  429.74    4851  429.26  4988.2  427.53  4996.4  426.64  5020.7  428.58
  5050.3  429.51  5257.9  429.61  5442.9   431.8    5569  434.21  5876.2  441.79
#Mann= 7 ,-1 , 0
  3318.6      .1       0  4471.4     .07       0  4479.2      .1       0
  5020.7     .05       0  5257.9      .1       0  5442.9     .05       0
    5569      .1       0
Bank Sta=4471.4,4479.2
XS Rating Curve= 0 ,0
Exp/Cntr=0.3,0.1

Type RM Length L Ch R = 1 ,5212    ,268,268,268
BEGIN DESCRIPTION:
UNT 030 in RCW 8.0
END DESCRIPTION:
XS GIS Cut Line= 3
       2017297.1     13457851.23      2017122.18     13458029.63
      2015229.62     13458843.55
#Sta/Elev= 30
  3649.7   460.4  3802.4   464.7  3899.5  463.64    3940  461.64  3977.3  458.28
  4024.3  450.64  4076.9  445.21  4190.4  437.06  4205.5  435.11    4229  428.67
    4258  425.89  4272.2   421.6  4272.8   420.8    4280   421.6  4288.4  426.49
  4299.2  428.18  4373.7  427.86    4680  426.28  4809.1  427.16  4974.1  427.92
  4995.9  423.14  5006.8  423.35  5028.6   427.6  5062.2  427.35  5213.1  427.43
  5406.5  428.16  5627.3  434.29  5732.2  440.81  5844.5  445.56  5959.7  444.67
#Mann= 9 ,-1 , 0
  3649.7      .1       0  4272.2      .1       0    4280      .1       0
  4373.7      .1       0  4809.1      .1       0  5062.2     .05       0
  5213.1      .1       0  5406.5      .1       0  5732.2      .1       0
#XS Ineff= 2 , 0
       0  4310.5     432               0
Permanent Ineff=
       F       F
Bank Sta=4974.1,5028.6
XS Rating Curve= 0 ,0
Exp/Cntr=0.3,0.1

Type RM Length L Ch R = 1 ,4944    ,430,430,430
BEGIN DESCRIPTION:
Mapping XS 1b90ead0
END DESCRIPTION:
XS GIS Cut Line= 3
      2017266.66     13457768.79      2016129.55      13458181.1
      2015023.75     13458740.51
#Sta/Elev= 30
  3607.5  456.02  3816.5  452.28  3877.8  448.49  4020.3  433.33  4162.4  427.91
  4193.4  422.21  4204.9  425.87  4259.9  426.83  4279.4  426.44  4310.6  420.94
    4322  423.63  4328.7  420.65  4329.3  419.85  4336.5  420.65  4346.5  421.67
  4353.9  426.47  4417.7  424.41  4449.6   420.8  4458.4  424.36  4481.5  425.96
  4599.2  425.42  4708.1  425.86  4971.6  426.62  4989.9   426.3  5001.5  426.74
  5139.3  426.06  5325.4  426.43  5686.8  439.56  5768.2  443.34  6056.3  442.47
#Mann= 9 ,-1 , 0
  3607.5      .1       0  4328.7     .07       0  4336.5      .1       0
  4599.2      .1       0  4708.1      .1       0  4989.9      .1       0
  5139.3      .1       0  5325.4      .1       0  5686.8      .1       0
#XS Ineff= 2 , 0
       0  4904.7     430               0
Permanent Ineff=
       F       F
Bank Sta=4971.6,5001.5
XS Rating Curve= 0 ,0
Exp/Cntr=0.3,0.1

Type RM Length L Ch R = 1 ,4514    ,437,437,437
BEGIN DESCRIPTION:
UNT 030 in RCW 7.0
END DESCRIPTION:
XS GIS Cut Line= 2
      2017084.43      13457642.9      2014976.19     13458360.15
#Sta/Elev= 30
  3443.2  446.74    3624  440.99  3706.7  442.39  3806.9  437.49  3963.7  435.84
  4052.5  426.93  4120.6  425.32  4146.7  422.01    4148   418.6  4148.6   417.8
  4155.8   418.6    4178  419.29  4183.3  422.53  4209.4  420.88  4255.9  425.12
  4287.6  424.69  4303.5  420.85  4360.9  424.44  4382.7  423.26    4429  425.14
  4692.3  425.85  4769.1  425.67  4988.3  424.98  5039.5  424.28  5082.4  424.91
  5193.2  429.33  5270.6   435.7  5460.1  434.24  5491.8  432.38  5670.1  438.77
#Mann= 7 ,-1 , 0
  3443.2      .1       0    4148     .07       0  4155.8      .1       0
  4692.3      .1       0  4769.1      .1       0  5039.5     .05       0
  5193.2      .1       0
#XS Ineff= 2 , 0
       0 4637.33     430               0
Permanent Ineff=
       F       F
Bank Sta=4988.3,5082.4
XS Rating Curve= 0 ,0
Exp/Cntr=0.3,0.1

Type RM Length L Ch R = 1 ,4077    ,194,194,194
BEGIN DESCRIPTION:
UNT 030 in RCW 6.0
END DESCRIPTION:
XS GIS Cut Line= 3
      2016780.64     13457399.84      2015716.68     13457708.14
      2015098.88     13457884.13
#Sta/Elev= 30
  3634.5  432.35  3779.9  430.26  3813.4   428.8    3859  428.32  3942.3  424.77
  4004.8  424.61  4056.8  427.11  4064.1  426.39  4069.3   427.1  4088.1  427.06
  4119.3  429.32  4136.5  429.14  4141.7  429.85  4181.8  424.11  4223.4  422.85
  4242.5  421.46  4254.6  418.43  4271.5   417.6  4272.2   416.8  4278.8   416.8
  4279.4   417.6  4286.4   420.2  4296.3  419.85    4320  422.61  4369.8  424.04
  4784.1  424.05    4973  423.05  5066.3  422.43  5079.7  423.26  5384.6  426.22
#Mann= 5 ,-1 , 0
  3634.5      .1       0  4271.5     .07       0  4279.4      .1       0
  4369.8      .1       0  4784.1      .1       0
#XS Ineff= 2 , 0
       0  4681.9     427               0
Permanent Ineff=
       F       F
Bank Sta=4973,5079.7
XS Rating Curve= 0 ,0
Exp/Cntr=0.3,0.1

Type RM Length L Ch R = 1 ,3883    ,181,181,181
BEGIN DESCRIPTION:
Mapping XS b734e61e
END DESCRIPTION:
XS GIS Cut Line= 2
      2016706.83     13457317.38      2014988.18      13457700.8
#Sta/Elev= 30
    3634  427.62  3827.6  424.29  3924.7  424.27  3963.1  422.66  3968.2  423.86
  3984.2  419.78  4016.8  417.59  4060.2  416.17  4103.7  417.61  4154.5  415.12
  4155.1  414.32  4162.4  415.12  4195.7  417.26  4200.8  416.27  4219.9  421.97
  4260.9  419.75  4301.1  420.82  4515.3  421.51  4537.5  423.78    4558  423.05
  4563.8  421.49    4569  422.68  4612.4  423.06  4655.9  422.09    4661  423.13
  4770.8  423.25  4883.4  421.66  4980.5   422.5  5029.3  422.42  5394.9  424.87
#Mann= 5 ,-1 , 0
    3634      .1       0  4154.5     .07       0  4162.4      .1       0
  4301.1      .1       0  4770.8      .1       0
#XS Ineff= 2 , 0
       0  4537.5     428               0
Permanent Ineff=
       F       F
Bank Sta=4980.5,5029.3
XS Rating Curve= 0 ,0
Exp/Cntr=0.3,0.1

Type RM Length L Ch R = 1 ,3702    ,317,317,317
BEGIN DESCRIPTION:
Mapping XS 0b2adbb8
END DESCRIPTION:
XS GIS Cut Line= 2
      2016641.67     13457239.27      2014979.91     13457604.84
#Sta/Elev= 30
  3637.3  425.13  3732.5  424.22  3951.3  424.28  4059.2  421.26    4103  420.34
  4135.6   420.4  4147.9  419.58  4148.5  418.78  4155.1  418.78  4155.8  419.58
  4156.9   420.7  4195.6  420.79  4200.7  421.36  4244.4  422.42  4293.3  422.49
  4337.1   421.5  4346.5  422.16  4371.1  421.81  4429.7  423.18  4688.3  423.06
    4849  421.84  4862.6  422.29  4985.4  421.61  5083.1  423.71  5098.1  423.68
  5126.9  422.18    5139  423.69  5169.8  424.36  5210.7  423.84  5338.8  423.89
#Mann= 5 ,-1 , 0
  3637.3      .1       0  4147.9     .07       0  4155.8      .1       0
  4346.5      .1       0  4688.3      .1       0
Bank Sta=4147.9,4155.8
XS Rating Curve= 0 ,0
Exp/Cntr=0.3,0.1

Type RM Length L Ch R = 1 ,3385    ,279,279,279
BEGIN DESCRIPTION:
UNT 030 in RCW 5.0
END DESCRIPTION:
XS GIS Cut Line= 3
      2016459.41     13457048.29      2015538.29     13457295.82
      2015052.24     13457440.06
#Sta/Elev= 30
  3975.8   422.7  4093.5  422.65  4218.6  421.03  4322.1  422.65  4408.2  422.29
  4482.9  419.02  4488.1  416.74  4504.4  416.18  4505.1  415.38  4511.9  415.38
  4512.5  416.18  4549.9  416.77  4570.6  421.43  4597.7  419.57  4622.4   420.9
  4643.1  420.55  4663.8  422.71  4717.6  421.67  4872.3  422.31  4964.3  421.47
  4979.7  421.04  4995.6  417.89    5006  420.22  5018.1  421.01    5151  421.93
    5246  424.06  5255.9  425.29  5266.8  424.13  5339.8  425.41  5436.6  425.46
#Mann= 3 ,-1 , 0
  3975.8      .1       0  4504.4     .07       0  4512.5      .1       0
Bank Sta=4504.4,4512.5
XS Rating Curve= 0 ,0
Exp/Cntr=0.3,0.1

Type RM Length L Ch R = 1 ,3106    ,348,348,348
BEGIN DESCRIPTION:
Mapping XS 7ae1e364
END DESCRIPTION:
XS GIS Cut Line= 2
      2016450.76     13456939.78      2015110.76     13457126.12
#Sta/Elev= 30
  3949.9  422.49  4046.6  422.34  4066.8  423.06  4187.9  420.82  4278.8  422.23
    4391  421.63  4462.7  418.26  4470.6  418.88  4480.7  418.19  4490.8  415.65
  4500.9  414.57  4541.3  416.78  4557.4   412.9  4558.1   412.1  4564.9   412.1
  4565.5   412.9  4571.6  414.76  4581.7  420.27  4591.8  421.27  4652.4  420.67
  4702.8  421.43  4854.3   421.3  4955.2  420.27  4975.4  419.75  4995.6  416.26
  5005.7  418.45  5025.9  418.67  5056.2  420.82  5217.7  424.34  5302.8  425.18
#Mann= 3 ,-1 , 0
  3949.9      .1       0  4557.4     .07       0  4565.5      .1       0
Bank Sta=4557.4,4565.5
XS Rating Curve= 0 ,0
Exp/Cntr=0.3,0.1

Type RM Length L Ch R = 1 ,2758    ,356,356,356
BEGIN DESCRIPTION:
Mapping XS 5c7c2744
END DESCRIPTION:
XS GIS Cut Line= 2
      2016342.26     13456718.43      2015075.63     13456855.28
#Sta/Elev= 30
  3958.3  424.07    4036  424.23  4146.6  422.93  4217.1  420.28  4247.2  420.28
  4257.3  419.73  4267.3  418.08  4277.4  418.19  4287.5  415.53  4297.5  415.64
  4307.6  418.94  4337.8  418.68  4344.1  416.43  4349.1  417.92  4357.9   412.7
  4363.9  412.52  4364.5  411.72  4371.3  411.72    4372  412.52    4378  416.37
    4388  419.34  4440.9  420.59  4569.1  419.47  4780.3  420.95  4961.4  417.78
  5001.8  415.47  5011.7  416.85  5061.9  420.27  5212.8  421.76  5232.3  421.09
#Mann= 3 ,-1 , 0
  3958.3      .1       0  4363.9     .07       0    4372      .1       0
Bank Sta=4363.9,4372
XS Rating Curve= 0 ,0
Exp/Cntr=0.3,0.1

Type RM Length L Ch R = 1 ,2402    ,170,170,170
BEGIN DESCRIPTION:
Mapping XS d5ed86b1
END DESCRIPTION:
XS GIS Cut Line= 2
      2016411.63     13456375.55      2015032.66     13456607.88
#Sta/Elev= 30
  3944.5  425.21  4022.2  425.41  4052.6  427.03  4083.1  425.09  4143.9  426.18
  4276.5  421.39  4316.3  417.69  4327.9  409.33  4328.6  408.53  4336.1  409.33
    4337  412.14  4377.1   416.7  4387.3  416.23  4392.5  413.19  4397.5  413.73
  4407.6   411.6    4438  416.82  4508.4  414.13  4610.4  414.49  4620.5  412.84
  4823.3  419.68  4924.8  417.71  4975.5  415.43  4985.6  414.42  4992.6  411.99
  5005.9  414.95    5016   415.3  5113.6  416.14    5229  420.12  5342.9  420.86
#Mann= 3 ,-1 , 0
  3944.5      .1       0  4327.9     .07       0  4336.1      .1       0
Bank Sta=4327.9,4336.1
XS Rating Curve= 0 ,0
Exp/Cntr=0.3,0.1

Type RM Length L Ch R = 1 ,2232    ,368,368,368
BEGIN DESCRIPTION:
UNT 030 in RCW 4.0
END DESCRIPTION:
XS GIS Cut Line= 3
      2016459.39     13456232.32        2015325.       13456425.
      2015009.56     13456402.18
#Sta/Elev= 30
  3825.1  423.82  4042.6  423.63  4235.3  419.25  4245.4  418.87  4265.7  412.23
  4284.9  409.97  4296.1  412.28  4302.2  408.61  4302.9  407.81  4310.4  408.61
  4316.4  412.77  4326.6  412.63  4345.2  418.19    4357  418.64  4397.6  417.03
  4417.9  411.89  4438.1  411.44  4458.4   414.3  4470.9  410.67  4488.9  412.45
    4499  415.17  4586.4  417.86    4712   419.2  4914.9  416.98  4985.8  413.96
  4995.8  411.47  5015.8   414.2  5035.9  414.03  5106.1   419.1    5292  423.71
#Mann= 3 ,-1 , 0
  3825.1      .1       0  4302.2     .07       0  4310.4      .1       0
Bank Sta=4302.2,4310.4
XS Rating Curve= 0 ,0
Exp/Cntr=0.3,0.1

Type RM Length L Ch R = 1 ,1864    ,332,332,332
BEGIN DESCRIPTION:
Mapping XS bf35f06a
END DESCRIPTION:
XS GIS Cut Line= 2
      2016350.91     13456136.83      2015091.26     13456148.25
#Sta/Elev= 30
  4089.3  422.61  4225.2  421.17  4305.2     418  4325.2  418.57  4425.2  415.81
  4434.5  414.41  4439.5  415.89  4445.2  414.06  4455.2  413.48  4465.2  415.38
  4475.2  414.34  4485.2  417.27  4495.2  417.32  4505.2  414.46  4541.1  407.59
  4541.8  406.79  4549.3  407.59  4575.2  410.94  4595.2  410.59  4605.2  408.91
  4625.2  409.24  4665.2  416.74  4695.2  417.67  4895.2  414.78  4985.2  410.31
  4995.3  408.91  5005.3  411.58  5015.3  412.25  5105.3  414.19    5349  422.58
#Mann= 3 ,-1 , 0
  4089.3      .1       0  4541.1     .07       0  4549.3      .1       0
Bank Sta=4541.1,4549.3
XS Rating Curve= 0 ,0
Exp/Cntr=0.3,0.1

Type RM Length L Ch R = 1 ,1532    ,139,139,139
BEGIN DESCRIPTION:
UNT 030 in RCW 3.0
END DESCRIPTION:
XS GIS Cut Line= 2
      2016168.58     13455828.68      2015059.99     13455937.31
#Sta/Elev= 30
  4198.4   420.2    4316  418.42  4342.7  413.74  4382.9   411.9  4412.5  411.89
  4417.5  410.64  4443.1  409.36  4463.2  412.08  4493.4  408.45    4519  409.46
  4524.1  408.51  4563.7  409.21  4583.8   407.9  4664.2  412.77  4754.6  414.32
  4823.6  411.49  4895.3  410.43  4955.6  411.66  4975.7  409.54  4985.7  407.02
  4991.7  406.97  4992.4  406.17  4999.2  406.17  4999.9  406.97  5005.8  409.63
  5031.6  411.15  5106.3  414.93  5138.1  414.93  5206.8  419.82  5312.3  423.67
#Mann= 3 ,-1 , 0
  4198.4      .1       0  4991.7     .07       0  4999.9      .1       0
Bank Sta=4991.7,4999.9
XS Rating Curve= 0 ,0
Exp/Cntr=0.3,0.1

Type RM Length L Ch R = 1 ,1393    ,395,395,395
BEGIN DESCRIPTION:
Mapping XS 8ae6b4ce
END DESCRIPTION:
XS GIS Cut Line= 3
      2016159.95     13455776.59      2015549.58     13455834.45
       2015099.5     13455745.99
#Sta/Elev= 30
  4194.5  419.17  4249.7  418.36  4279.8  416.64    4310  417.57  4335.9  415.25
  4444.1  410.31  4470.7   414.7 4486.36409.8073  4510.9  407.21    4541  408.13
  4547.3  410.48  4561.1   409.1  4581.2  414.07  4591.2  411.44  4601.3  410.45
  4763.7  414.18  4863.2  411.58  4944.8  412.46  4975.3  411.27  4983.3  409.42
  4988.4  410.68  4991.6   405.5  4992.3   404.7  4999.9   405.5  5005.9  408.25
 5041.15409.8063  5056.9  411.66  5142.6  413.18  5199.5  418.16  5266.3  421.47
#Mann= 3 ,-1 , 0
  4194.5      .1       0  4991.6     .07       0  4999.9      .1       0
Bank Sta=4486.36,5041.15
XS Rating Curve= 0 ,0
Exp/Cntr=0.3,0.1

Type RM Length L Ch R = 1 ,998     ,319,319,319
BEGIN DESCRIPTION:
UNT 030 in RCW 2.0
END DESCRIPTION:
XS GIS Cut Line= 4
      2015916.29     13455495.14      2015599.27     13455608.97
      2015347.97     13455467.04      2015182.43     13455530.41
#Sta/Elev= 30
  4506.9  420.31  4548.2  419.73  4561.4  417.39  4609.6  413.41  4696.5  410.01
  4710.2  408.54  4727.3  409.15 4738.14408.2283  4773.9  404.56  4795.2  407.24
  4805.8  410.27  4837.7  406.77  4858.2  407.87  4871.6  407.08  4907.2  411.01
  4923.1  409.06  4960.7  408.88  4982.4  406.51  4993.8  404.13  4994.5  403.33
  5002.1  404.13 5003.84408.2323  5019.9  412.19    5069  410.19  5136.5  411.88
  5170.8  413.65  5195.5  416.51  5200.8  415.66  5220.2  417.33  5309.6  418.49
#Mann= 3 ,-1 , 0
  4506.9      .1       0  4993.8     .07       0  5002.1      .1       0
Bank Sta=4738.14,5003.84
XS Rating Curve= 0 ,0
Exp/Cntr=0.3,0.1
