--- UNT 059 in RCW.prj (project) ---

Proj Title=UNT 059 in RCW Base Level Engineering
Current Plan=p01
Default Exp/Contr=0.3,0.1
English Units
Geom File=g01
Flow File=f01
Plan File=p01
Y Axis Title=Elevation
X Axis Title(PF)=Main Channel Distance
X Axis Title(XS)=Station
BEGIN DESCRIPTION:
UNT 059 in RCW
END DESCRIPTION:
DSS Export Rating Curves= 0
DSS Export Rating Curve Sorted= 0
DSS Export Volume Flow Curves= 0
DXF OffsetX= 0
DXF OffsetY= 0
DXF ScaleX= 1
DXF ScaleY= 10

--- UNT 059 in RCW.p01 (plan) ---

Plan Title=Multiple Run
Short Identifier=Multiple
Geom File=g01
Flow File=f01
Subcritical Flow
K Sum by GR= 0
Std Step Tol= 0.01
Critical Tol= 0.01
Num of Std Step Trials= 20
Max Error Tol= 0.3
Flow Tol Ratio= 0.001
Split Flow NTrial= 30
Split Flow Tol= 0.02
Split Flow Ratio= 0.02
Log Output Level= 0
Friction Slope Method= 1
Unsteady Friction Slope Method= 2
Unsteady Bridges Friction Slope Method= 1
Parabolic Critical Depth
Global Vel Dist=  1 , 1 , 1
Global Log Level= 0
CheckData=True
Encroach Param= -1, 0, 0, 0
BEGIN DESCRIPTION:
Multiple Run
END DESCRIPTION:

--- UNT 059 in RCW.f01 (steady flow) ---

Flow Title=Multiple
Program Version=5.05
Number of Profiles= 7
Profile Names=10-year,25-year,50-year,1pct_min,100-year,1pct_plu,500-year
River Rch & RM=UNT 059 in RCW,Reach-1         ,28263
     160     218     264     160     320     638     475
River Rch & RM=UNT 059 in RCW,Reach-1         ,27192
     278     389     481     297     592    1180     909
River Rch & RM=UNT 059 in RCW,Reach-1         ,20991
     339     476     592     366     730    1457    1130
River Rch & RM=UNT 059 in RCW,Reach-1         ,16641
     395     558     695     431     859    1715    1336
River Rch & RM=UNT 059 in RCW,Reach-1         ,13730
     546     780     980     611    1219    2432    1919
River Rch & RM=UNT 059 in RCW,Reach-1         ,12549
     546     780     980     611    1219    2432    1919
Boundary for River Rch & Prof#=UNT 059 in RCW,Reach-1         , 1
Up Type= 0
Dn Type= 3
Dn Slope=0.005
Boundary for River Rch & Prof#=UNT 059 in RCW,Reach-1         , 2
Up Type= 0
Dn Type= 3
Dn Slope=0.005
Boundary for River Rch & Prof#=UNT 059 in RCW,Reach-1         , 3
Up Type= 0
Dn Type= 3
Dn Slope=0.005
Boundary for River Rch & Prof#=UNT 059 in RCW,Reach-1         , 4
Up Type= 0
Dn Type= 3
Dn Slope=0.005
Boundary for River Rch & Prof#=UNT 059 in RCW,Reach-1         , 5
Up Type= 0
Dn Type= 3
Dn Slope=0.005
Boundary for River Rch & Prof#=UNT 059 in RCW,Reach-1         , 6
Up Type= 0
Dn Type= 3
Dn Slope=0.005
Boundary for River Rch & Prof#=UNT 059 in RCW,Reach-1         , 7
Up Type= 0
Dn Type= 3
Dn Slope=0.005
DSS Import GetInterval= 0
DSS Import GetPeak= 0
DSS Import FillOption= 0

--- UNT 059 in RCW.g01 (geometry) ---

Geom Title=Existing Conditions

River Reach=UNT 059 in RCW,Reach-1
Reach XY= 30
      2050020.80     13415814.54      2051080.80     13416394.54
      2052184.57     13418342.20      2051919.81     13419249.31
      2052083.66     13419655.13      2051850.37     13419761.47
      2052033.74     13420339.81      2051750.80     13420754.54
      2053080.80     13421144.54      2053590.80     13421614.54
      2054260.80     13423024.54      2055078.39     13423370.16
      2057255.15     13423454.98      2058161.43     13423000.95
      2058070.80     13423474.54      2058410.80     13423654.54
      2058650.80     13423444.54      2058820.80     13424094.54
      2059180.80     13423934.54      2059010.80     13423384.54
      2059510.80     13423464.54      2059540.80     13423694.54
      2060200.80     13423874.54      2060100.80     13424634.54
      2060460.80     13425024.54      2061020.80     13424984.54
      2061880.80     13425834.54      2062450.80     13425504.54
      2062990.80     13426224.54      2063780.80     13426264.54

Type RM Length L Ch R = 1,28263,523,523,523
BEGIN DESCRIPTION:
UNT 059 in RCW 30.0
END DESCRIPTION:
XS GIS Cut Line= 3
      2049575.00     13416525.00      2050085.14     13415932.29
      2050668.32     13414229.62
#Sta/Elev= 30
  4167.5  428.46  4238.3  425.27  4309.7  423.14  4472.0  418.35  4564.2  416.45
  4699.1  414.53  4854.9  414.17  4957.2  413.15  4985.9  411.49  4986.4  410.69
  4991.4  410.69  4991.9  411.49  5000.1  411.59  5031.4  414.22  5119.9  413.23
  5207.0  414.76  5395.5  417.60  5552.7  420.41  5654.9  423.93  5703.8  424.15
  5740.4  425.25  5766.4  427.02  5898.0  430.74  6110.5  434.09  6167.8  436.60
  6230.4  437.56  6287.7  440.00  6444.1  443.78  6626.5  442.38  6749.3  439.02
#Mann=6,-1,0
  4167.5     0.1       0  4309.7    0.05       0  4985.9    0.07       0
  4991.9    0.05       0  5207.0    0.05       0  5395.5     0.1       0
Bank Sta=4985.9,4991.9
Exp/Cntr=0.3,0.1

Type RM Length L Ch R = 1,27740,548,548,548
BEGIN DESCRIPTION:
UNT 059 in RCW 29.0
END DESCRIPTION:
XS GIS Cut Line= 3
      2049757.05     13416802.05      2051132.02     13415463.54
      2050975.77     13413921.83
#Sta/Elev= 30
  3952.5  425.96  3991.5  426.32  4161.0  421.08  4237.5  419.49  4422.8  415.13
  4585.4  412.56  4961.7  411.35  4992.7  409.77  4993.2  408.97  4998.2  408.97
  4998.7  409.77  5023.9  410.79  5073.4  411.23  5144.1  411.28  5193.5  410.53
  5335.0  412.66  5370.4  412.19  5533.0  412.94  5568.5  412.55  5667.3  414.46
  5888.2  415.19  6092.9  418.28  6201.6  420.88  6804.7  424.48  6886.6  426.25
  6945.4  426.95  6975.6  426.63  6995.7  427.43  7307.2  431.14  7421.0  433.42
#Mann=5,-1,0
  3952.5     0.1       0  4237.5    0.05       0  4961.7     0.1       0
  4992.7    0.07       0  4998.7     0.1       0
Bank Sta=4992.7,4998.7
Exp/Cntr=0.3,0.1

Type RM Length L Ch R = 1,27192,442,442,442
BEGIN DESCRIPTION:
UNT 059 in RCW 28.0
END DESCRIPTION:
XS GIS Cut Line= 3
      2050025.01     13416824.99      2050925.00     13416325.00
      2052090.15     13414896.07
#Sta/Elev= 30
  3966.0  425.03  4120.4  420.43  4239.4  415.18  4332.1  412.74  4503.6  410.06
  4965.8  409.37  4992.7  407.44  5009.2  407.46  5020.0  408.38  5066.6  409.58
  5121.1  406.83  5121.6  406.03  5126.6  406.03  5127.1  406.83  5188.0  408.49
  5563.5  410.70  5827.1  413.00  5855.8  413.83  5983.6  414.43  5990.0  413.43
  6018.8  412.89  6054.0  414.09  6076.2  413.58  6140.1  414.41  6288.8  419.09
  6331.9  419.77  6651.4  431.80  6729.6  433.42  6758.4  433.11  6839.3  436.12
#Mann=5,-1,0
  3966.0     0.1       0  4120.4    0.05       0  5020.0     0.1       0
  5121.1    0.03       0  5127.1     0.1       0
Bank Sta=5121.1,5127.1
Exp/Cntr=0.3,0.1

Type RM Length L Ch R = 1,26750,426,426,426
BEGIN DESCRIPTION:
UNT 059 in RCW 27.0
END DESCRIPTION:
XS GIS Cut Line= 3
      2050125.04     13416974.99      2051225.00     13416575.00
      2052538.25     13415312.52
#Sta/Elev= 30
  3855.9  423.98  4004.8  420.41  4131.1  415.57  4228.3  412.77  4441.1  409.26
  4721.1  407.05  4909.3  406.75  4955.2  407.44  4980.4  406.41  4985.8  404.80
  4993.9  404.61  5007.9  403.65  5008.4  402.85  5013.7  402.85  5014.2  403.65
  5029.8  404.96  5040.3  406.78  5054.5  406.92  5125.2  406.91  5153.5  405.16
  5189.1  406.58  5556.7  409.04  5705.4  408.98  5825.5  410.71  5945.7  413.66
  6143.8  423.31  6476.2  429.55  6681.2  436.10  6773.3  438.13  6848.0  441.01
#Mann=5,-1,0
  3855.9     0.1       0  4131.1    0.05       0  4993.9     0.1       0
  5007.9    0.07       0  5014.2     0.1       0
Bank Sta=5007.9,5014.2
Exp/Cntr=0.3,0.1

Type RM Length L Ch R = 1,26324,410,410,410
BEGIN DESCRIPTION:
UNT 059 in RCW 26.0
END DESCRIPTION:
XS GIS Cut Line= 3
      2050325.00     13417125.00      2051425.00     13416925.00
      2052745.68     13415839.30
#Sta/Elev= 30
  3856.2  421.00  4048.0  416.03  4111.6  412.78  4181.5  412.23  4335.2  408.93
  4447.0  407.71  4466.0  407.00  4842.1  405.44  4944.4  404.36  4977.5  403.45
  4999.1  401.78  4999.6  400.98  5004.9  400.98  5005.4  401.78  5024.4  404.13
  5038.8  405.17  5080.4  404.46  5144.3  404.57  5173.0  403.56  5201.7  404.58
  5272.0  405.48  5500.1  405.80  5621.4  407.33  5720.4  409.48  5755.6  409.51
  5912.0  412.87  6082.7  414.71  6217.0  418.16  6274.3  418.85  6683.9  430.04
#Mann=4,-1,0
  3856.2    0.05       0  4944.4     0.1       0  4999.1    0.07       0
  5005.4     0.1       0
Bank Sta=4999.1,5005.4
Exp/Cntr=0.3,0.1

Type RM Length L Ch R = 1,25914,299,299,299
BEGIN DESCRIPTION:
UNT 059 in RCW 25.0
END DESCRIPTION:
XS GIS Cut Line= 3
      2050559.10     13417520.83      2051675.00     13417225.00
      2052740.73     13416526.48
#Sta/Elev= 30
  3861.0  416.40  3943.5  414.82  4174.4  407.22  4289.8  405.54  4445.4  404.41
  4901.7  403.71  4984.3  403.05  5001.9  400.63  5002.4  399.83  5007.8  399.83
  5008.3  400.63  5018.4  400.81  5023.0  402.06  5044.1  403.52  5074.3  403.44
  5095.4  402.06  5110.5  401.88  5131.5  403.06  5137.5  404.00  5152.6  404.46
  5218.7  402.48  5267.1  403.34  5390.7  403.17  5659.1  404.84  5773.6  407.16
  5912.2  412.94  6011.7  417.98  6105.2  421.46  6249.9  421.78  6289.7  421.30
#Mann=4,-1,0
  3861.0    0.05       0  4984.3     0.1       0  5001.9    0.07       0
  5008.3     0.1       0
Bank Sta=5001.9,5008.3
Exp/Cntr=0.3,0.1

Type RM Length L Ch R = 1,25615,211,211,211
BEGIN DESCRIPTION:
Mapping XS f47b9d48
END DESCRIPTION:
XS GIS Cut Line= 4
      2050874.56     13417595.36      2051512.54     13417591.02
      2052055.08     13417343.63      2052745.19     13416636.15
#Sta/Elev= 30
  4106.1  407.10  4166.5  405.24  4346.5  403.51  4516.6  402.76  4767.0  403.01
  4931.8  401.86  4977.6  402.56  4996.4  400.04  4996.9  399.24  5002.3  399.24
  5002.8  400.04  5036.9  402.23  5129.1  401.60  5155.5  401.97  5180.7  402.75
  5263.4  402.08  5329.9  402.24  5388.9  401.25  5424.1  401.91  5558.6  402.45
  5685.9  404.34  5707.1  405.13  5841.4  406.37  5905.1  408.13  5975.8  411.58
  6039.4  413.41  6060.7  414.75  6103.1  416.08  6244.6  419.30  6328.7  419.75
#Mann=5,-1,0
  4106.1    0.05       0  4931.8    0.12       0  4996.4    0.07       0
  5002.8    0.12       0  5155.5     0.1       0
Bank Sta=4996.4,5002.8
Exp/Cntr=0.3,0.1

Type RM Length L Ch R = 1,25404,225,225,225
BEGIN DESCRIPTION:
Mapping XS 42e81434
END DESCRIPTION:
XS GIS Cut Line= 4
      2050731.30     13417660.47      2051621.05     13417677.83
      2052068.10     13417621.40      2052797.24     13416709.98
#Sta/Elev= 30
  3852.6  410.99  3916.3  409.49  4056.3  404.81  4186.4  403.31  4586.4  402.66
  4766.7  401.74  4796.9  402.11  4882.1  400.89  4899.8  400.58  4978.3  402.00
  5005.4  399.80  5005.9  399.00  5011.3  399.00  5011.8  399.80  5044.2  401.80
  5059.0  401.29  5098.6  401.45  5179.9  401.20  5245.2  400.19  5301.1  401.11
  5466.1  401.17  5565.3  402.83  5771.8  405.11  5864.7  407.16  5935.1  409.59
  5970.3  409.26  6042.3  410.42  6156.0  413.39  6319.3  416.11  6360.3  417.64
#Mann=7,-1,0
  3852.6    0.05       0  4882.1     0.1       0  4899.8    0.12       0
  5005.4    0.07       0  5011.8    0.12       0  5098.6    0.05       0
  5301.1     0.1       0
Bank Sta=5005.4,5011.8
Exp/Cntr=0.3,0.1

Type RM Length L Ch R = 1,25179,185,185,185
BEGIN DESCRIPTION:
Mapping XS 473c4963
END DESCRIPTION:
XS GIS Cut Line= 4
      2049975.82     13417677.09      2051199.73     13417880.20
      2052574.73     13417854.16      2053261.08     13417505.79
#Sta/Elev= 30
  3046.6  414.44  3355.0  411.81  3394.6  411.96  3704.7  412.96  4018.9  403.76
  4129.0  402.67  4402.5  402.08  4452.6  398.77  4489.3  398.51  4489.8  397.71
  4495.4  397.71  4495.9  398.51  4572.6  402.02  4612.6  399.86  4662.6  399.05
  4902.6  399.86  5085.4  398.97  5272.7  399.62  5349.9  398.80  5432.7  399.95
  5492.7  398.70  5611.2  398.94  5720.2  404.14  5797.4  404.98  5935.3  408.62
  6113.0  415.52  6178.8  418.00  6257.2  419.59  6369.3  423.88  6432.2  427.41
#Mann=12,-1,0
  3046.6    0.05       0  3355.0     0.1       0  3394.6    0.05       0
  4129.0     0.1       0  4489.3    0.07       0  4495.9     0.1       0
  5085.4    0.07       0  5349.9     0.1       0  5611.2    0.05       0
  5935.3     0.1       0  6113.0    0.05       0  6178.8     0.1       0
Bank Sta=4489.3,4495.9
Exp/Cntr=0.3,0.1

Type RM Length L Ch R = 1,24994,817,817,817
BEGIN DESCRIPTION:
Mapping XS c176202d
END DESCRIPTION:
XS GIS Cut Line= 4
      2049845.54     13417812.49      2050751.81     13418109.37
      2052559.10     13418010.41      2053460.07     13417593.78
#Sta/Elev= 30
  2828.1  414.07  2945.3  412.82  3322.1  409.01  3622.6  409.22  3951.7  401.70
  4045.3  400.66  4202.8  400.36  4926.7  399.39  4993.5  397.92  4994.0  397.12
  4999.6  397.12  5000.1  397.92  5096.9  399.14  5347.3  398.35  5467.5  399.26
  5653.3  401.82  5730.3  403.54  5735.8  404.38  5764.3  405.07  5867.7  406.05
  5970.6  408.25  6090.8  413.14  6165.1  415.29  6171.2  416.03  6308.2  420.95
  6422.8  426.66  6520.1  430.11  6525.6  429.67  6565.9  430.77  6584.4  432.05
#Mann=6,-1,0
  2828.1    0.05       0  2945.3     0.1       0  4202.8    0.05       0
  4993.5    0.03       0  5000.1    0.05       0  5867.7     0.1       0
Bank Sta=4993.5,5000.1
Exp/Cntr=0.3,0.1

Type RM Length L Ch R = 1,24177,1052,1052,1052
BEGIN DESCRIPTION:
UNT 059 in RCW 22.0
END DESCRIPTION:
XS GIS Cut Line= 3
      2049984.42     13418708.33      2052536.53     13418769.09
      2053578.19     13418300.35
#Sta/Elev= 30
  2774.3  406.88  3215.0  403.51  3445.1  403.00  3855.2  399.17  3975.2  397.27
  4005.2  397.78  4085.2  397.33  4155.3  395.94  4275.3  396.59  4405.3  395.55
  4545.4  396.45  4585.4  395.84  4666.4  395.97  4942.8  395.28  5002.2  393.47
  5002.7  392.67  5008.4  392.67  5008.9  393.47  5025.5  394.83  5045.5  395.49
  5125.5  394.74  5155.6  395.37  5285.6  394.88  5424.5  395.86  5593.5  396.63
  5668.5  398.18  5807.4  399.69  5972.4  406.11  6268.5  412.23  6469.4  417.54
#Mann=5,-1,0
  2774.3     0.1       0  4666.4    0.05       0  5002.2    0.03       0
  5008.9    0.05       0  5424.5     0.1       0
Bank Sta=5002.2,5008.9
Exp/Cntr=0.3,0.1

Type RM Length L Ch R = 1,23125,552,552,552
BEGIN DESCRIPTION:
Mapping XS 73ccbfc1
END DESCRIPTION:
XS GIS Cut Line= 4
      2050562.06     13418906.14      2051733.90     13419470.36
      2052246.05     13419613.59      2053339.81     13418545.87
#Sta/Elev= 30
  3328.4  402.37  3620.2  400.37  3908.4  395.83  4185.4  393.35  4394.6  392.84
  4490.7  391.82  4552.5  392.24  4581.2  391.56  4640.5  392.38  4879.3  393.03
  4972.8  392.70  5004.0  391.26  5045.5  392.99  5074.2  392.41  5229.7  391.93
  5254.6  391.24  5255.1  390.44  5260.8  390.44  5261.3  391.24  5300.4  392.18
  5458.3  391.78  5583.3  391.53  5767.2  393.31  6014.7  393.33  6099.5  394.57
  6290.6  395.81  6333.0  396.95  6368.3  399.09  6516.7  405.48  6689.3  409.77
#Mann=5,-1,0
  3328.4     0.1       0  5074.2    0.05       0  5254.6    0.07       0
  5261.3    0.05       0  5458.3     0.1       0
Bank Sta=5254.6,5261.3
Exp/Cntr=0.3,0.1

Type RM Length L Ch R = 1,22573,367,367,367
BEGIN DESCRIPTION:
UNT 059 in RCW 21.0
END DESCRIPTION:
XS GIS Cut Line= 4
      2049925.00     13419275.00      2050998.34     13419991.32
      2052519.17     13419803.82      2053474.98     13418475.03
#Sta/Elev= 30
  2762.3  407.63  3310.5  400.87  3526.8  399.69  3722.1  396.06  4220.6  392.35
  4432.2  389.90  4613.6  389.82  4637.2  389.12  4684.1  390.28  4734.5  389.85
  4915.9  391.48  4966.9  390.99  5013.3  388.57  5013.8  387.77  5019.5  387.77
  5020.0  388.57  5043.0  390.36  5067.0  390.76  5212.4  391.04  5512.7  389.97
  5774.7  389.90  5831.2  389.06  5881.5  390.60  5982.2  391.36  6411.8  391.91
  6441.2  392.82  6548.0  393.28  6678.1  395.69  6921.2  406.53  7221.9  413.15
#Mann=5,-1,0
  2762.3     0.1       0  5013.3    0.07       0  5020.0     0.1       0
  5212.4    0.05       0  5512.7     0.1       0
Bank Sta=5013.3,5020
Exp/Cntr=0.3,0.1

Type RM Length L Ch R = 1,22206,1215,1215,1215
BEGIN DESCRIPTION:
Mapping XS db28e155
END DESCRIPTION:
XS GIS Cut Line= 4
      2049296.97     13420588.54      2051366.39     13420387.15
      2052553.89     13419998.26      2053435.84     13418755.21
#Sta/Elev= 30
  2221.3  405.65  2631.3  401.47  2681.5  400.74  2719.5  398.17  2802.1  397.31
  2952.8  400.91  3013.1  399.23  3495.3  395.00  4319.1  390.61  4499.0  388.87
  4517.4  387.16  4517.9  386.36  4524.1  387.16  4572.6  388.66  4642.9  387.44
  4667.3  388.78  4871.1  389.87  4972.5  389.49  5004.0  387.43  5046.1  389.89
  5108.9  389.50  5401.1  388.69  5575.2  387.46  5896.0  390.31  6011.2  390.01
  6320.7  390.55  6671.3  393.33  6801.7  396.94  7009.6  405.67  7074.2  406.94
#Mann=7,-1,0
  2221.3     0.1       0  4517.4    0.07       0  4524.1     0.1       0
  5108.9    0.05       0  5401.1     0.1       0  5896.0    0.05       0
  6011.2     0.1       0
Bank Sta=4517.4,4524.1
Exp/Cntr=0.3,0.1

Type RM Length L Ch R = 1,20991,452,452,452
BEGIN DESCRIPTION:
UNT 059 in RCW 20.0
END DESCRIPTION:
XS GIS Cut Line= 3
      2050875.03     13421574.98      2052075.00     13420875.00
      2053474.99     13418875.01
#Sta/Elev= 30
  3627.4  399.87  4014.8  398.72  4388.6  388.79  4774.4  386.89  4819.8  386.80
  4848.3  384.60  4900.8  384.98  4935.6  386.97  4983.2  384.54  4983.9  383.74
  4990.7  383.74  4991.3  384.54  5202.8  386.72  5330.0  386.91  5487.7  387.10
  5699.7  387.39  5813.1  386.52  5914.2  388.04  5943.9  387.04  5979.6  388.18
  6221.4  389.34  6584.0  389.39  6920.4  391.83  6956.1  390.93  7018.9  392.69
  7114.0  392.99  7134.9  394.41  7221.2  396.50  7313.6  400.78  7457.9  404.68
#Mann=8,-1,0
  3627.4    0.05       0  4774.4     0.1       0  4983.2    0.07       0
  4991.3     0.1       0  5330.0    0.05       0  5487.7     0.1       0
  6221.4    0.05       0  6584.0     0.1       0
Bank Sta=4983.2,4991.3
Exp/Cntr=0.3,0.1

Type RM Length L Ch R = 1,20539,421,421,421
BEGIN DESCRIPTION:
UNT 059 in RCW 19.0
END DESCRIPTION:
XS GIS Cut Line= 3
      2050875.02     13422524.98      2052475.00     13420975.00
      2053475.00     13418975.00
#Sta/Elev= 30
  2767.7  407.49  2841.9  406.30  2858.8  406.02  2964.9  403.30  3269.7  396.31
  3800.4  389.57  4111.3  386.46  4295.3  385.43  4578.0  385.82  4726.2  383.90
  4761.9  384.45  4811.5  383.21  4945.8  384.93  4960.0  384.27  4984.2  380.76
  4984.9  379.96  4992.3  380.76  5017.7  384.15  5031.7  384.75  5107.1  384.00
  5241.3  385.60  5434.2  385.19  5713.9  386.83  5898.1  388.01  6337.0  388.21
  6591.9  390.11  6814.9  391.42  6865.2  392.64  6887.6  392.02  7231.4  402.64
#Mann=10,-1,0
  2767.7    0.08       0  2841.9    0.05       0  2858.8    0.08       0
  2964.9     0.1       0  3800.4    0.05       0  4726.2     0.1       0
  4984.2    0.07       0  4992.3     0.1       0  5713.9    0.05       0
  6591.9     0.1       0
Bank Sta=4984.2,4992.3
Exp/Cntr=0.3,0.1

Type RM Length L Ch R = 1,20118,473,473,473
BEGIN DESCRIPTION:
UNT 059 in RCW 18.0
END DESCRIPTION:
XS GIS Cut Line= 3
      2051174.98     13422675.02      2052775.00     13421125.00
      2053575.01     13419124.97
#Sta/Elev= 30
  2752.1  405.00  2891.3  402.26  2998.5  399.51  3353.2  391.83  3388.7  390.20
  3467.3  388.65  3586.7  386.67  3911.9  385.68  4138.2  383.42  4315.0  384.67
  4742.5  383.67  4824.3  382.67  4951.6  383.82  4965.8  383.38  4976.3  380.91
  4982.5  380.91  4989.2  379.48  4997.2  378.98  4997.9  378.18  5004.7  378.18
  5005.5  378.98  5048.5  383.00  5383.4  384.71  5689.3  386.26  6262.8  387.66
  6565.7  389.91  6627.7  389.66  6789.2  391.97  6825.6  391.84  7133.9  400.24
#Mann=9,-1,0
  2752.1    0.08       0  2891.3    0.05       0  2998.5     0.1       0
  3467.3    0.05       0  4742.5     0.1       0  4997.2    0.07       0
  5005.5     0.1       0  5383.4    0.05       0  6565.7     0.1       0
Bank Sta=4997.2,5005.5
Exp/Cntr=0.3,0.1

Type RM Length L Ch R = 1,19645,529,529,529
BEGIN DESCRIPTION:
UNT 059 in RCW 17.0
END DESCRIPTION:
XS GIS Cut Line= 3
      2051524.98     13422775.02      2053125.00     13421225.00
      2053925.01     13419224.97
#Sta/Elev= 30
  2752.1  400.61  2858.2  396.73  3197.7  387.74  3482.6  384.07  3834.2  382.56
  4215.9  383.35  4357.4  382.40  4433.9  382.90  4604.9  383.05  4682.8  381.54
  4718.1  382.20  4958.6  382.49  4989.2  381.13  5014.7  379.10  5015.4  378.30
  5022.3  378.30  5023.0  379.10  5024.2  379.85  5055.2  382.15  5356.8  384.00
  5732.1  384.88  6350.1  387.23  6478.2  388.28  6573.8  389.95  6801.3  396.32
  6820.2  395.83  6903.6  397.35  7004.6  397.46  7065.2  399.19  7133.9  400.07
#Mann=7,-1,0
  2752.1     0.1       0  3482.6    0.05       0  4433.9     0.1       0
  5014.7    0.07       0  5023.0     0.1       0  5732.1    0.05       0
  6350.1     0.1       0
Bank Sta=5014.7,5023
Exp/Cntr=0.3,0.1

Type RM Length L Ch R = 1,19116,631,631,631
BEGIN DESCRIPTION:
UNT 059 in RCW 16.0
END DESCRIPTION:
XS GIS Cut Line= 3
      2051774.97     13422775.02      2053375.00     13421525.00
      2053975.00     13419725.00
#Sta/Elev= 30
  2948.0  395.17  3297.1  384.65  3468.3  382.38  3703.2  381.15  4088.5  382.61
  4387.0  381.72  4508.9  380.36  4614.9  380.90  4635.8  379.78  4658.3  381.02
  4728.8  381.20  4772.2  379.48  4822.0  379.08  4886.2  380.96  4907.0  380.71
  4921.5  377.39  4956.7  378.76  4984.8  376.89  4985.5  376.09  4992.4  376.09
  4993.1  376.89  4999.5  378.33  5031.1  380.25  5104.9  381.37  6027.5  384.53
  6201.2  384.56  6416.9  386.12  6633.4  389.18  6780.9  393.77  6875.8  394.95
#Mann=5,-1,0
  2948.0     0.1       0  4984.8    0.07       0  4993.1     0.1       0
  6027.5    0.05       0  6416.9     0.1       0
Bank Sta=4984.8,4993.1
Exp/Cntr=0.3,0.1

Type RM Length L Ch R = 1,18485,689,689,689
BEGIN DESCRIPTION:
Mapping XS 7d6f5338
END DESCRIPTION:
XS GIS Cut Line= 4
      2052923.20     13422150.34      2053381.50     13422105.20
      2054006.50     13421563.54      2054072.27     13420968.13
#Sta/Elev= 30
  4220.5  381.38  4453.4  378.53  4534.4  378.88  4564.0  377.60  4604.1  379.00
  4704.9  379.09  4790.4  378.20  4839.7  378.69  4903.4  377.78  4917.6  378.54
  4938.5  378.21  4946.1  377.40  4952.7  378.26  4960.4  377.44  4967.0  377.91
  4974.6  376.42  4991.3  375.42  4992.0  374.62  4998.9  374.62  4999.7  375.42
  5016.5  377.33  5066.7  379.09  5151.2  379.22  5208.2  378.12  5257.6  379.25
  5297.8  378.97  5508.1  378.56  5748.1  380.38  5919.1  380.36  6107.1  381.45
#Mann=4,-1,0
  4220.5     0.1       0  4991.3    0.07       0  4999.7     0.1       0
  5297.8    0.05       0
Bank Sta=4991.3,4999.7
Exp/Cntr=0.3,0.1

Type RM Length L Ch R = 1,17796,524,524,524
BEGIN DESCRIPTION:
Mapping XS ee61b31c
END DESCRIPTION:
XS GIS Cut Line= 4
      2052881.49     13422601.73      2053534.28     13422532.29
      2054107.19     13422171.18      2054183.42     13421488.62
#Sta/Elev= 30
  3977.9  379.14  4031.7  378.45  4087.9  379.01  4132.3  378.30  4333.4  378.79
  4413.9  377.99  4514.4  377.87  4615.0  376.58  4676.4  377.52  4812.9  377.54
  4895.3  376.11  4916.5  374.81  4966.2  375.54  4974.2  375.25  4989.5  373.29
  4991.2  372.49  4991.9  371.69  4998.8  371.69  4999.6  372.49  5037.8  376.52
  5089.5  377.38  5151.2  376.39  5277.9  377.12  5378.2  376.35  5520.6  376.29
  5589.5  377.02  5605.9  377.67  5639.8  377.30  5871.2  378.91  5998.4  379.12
#Mann=4,-1,0
  3977.9     0.1       0  4991.2    0.07       0  4999.6     0.1       0
  5151.2    0.05       0
Bank Sta=4991.2,4999.6
Exp/Cntr=0.3,0.1

Type RM Length L Ch R = 1,17272,631,631,631
BEGIN DESCRIPTION:
Mapping XS fa017a76
END DESCRIPTION:
XS GIS Cut Line= 3
      2053596.77     13422952.43      2054204.42     13422549.65
      2054207.89     13421632.97
#Sta/Elev= 30
  4435.5  385.65  4439.6  385.73  4445.6  383.18  4454.7  383.27  4460.7  380.45
  4473.6  380.36  4475.7  380.34  4481.7  377.67  4577.3  373.96  4605.1  375.92
  4635.2  376.76  4671.3  375.23  4821.6  376.14  4966.0  374.38  4991.9  371.74
  4992.7  370.94  4999.6  370.94  5000.3  371.74  5053.3  375.44  5059.3  373.41
  5068.3  374.30  5074.3  373.17  5089.4  375.48  5143.7  375.61  5309.2  374.97
  5489.2  376.39  5659.2  376.29  5679.2  375.61  5839.2  377.52  6081.2  378.69
#Mann=5,-1,0
  4435.5    0.05       0  4473.6     0.1       0  4991.9    0.07       0
  5000.3     0.1       0  5143.7    0.05       0
Bank Sta=4991.9,5000.3
Exp/Cntr=0.3,0.1

Type RM Length L Ch R = 1,16641,53,53,53
BEGIN DESCRIPTION:
Mapping XS 9c3fb150
END DESCRIPTION:
XS GIS Cut Line= 3
      2053934.43     13423258.54      2054432.68     13422685.64
      2054282.51     13421734.27
#Sta/Elev= 30
  4602.8  390.05  4733.3  386.36  4761.8  384.43  4811.1  382.62  4853.9  379.66
  4860.5  379.73  4868.1  378.70  4874.8  378.99  4882.4  378.07  4917.5  377.05
  4946.0  374.62  4974.5  374.17  5009.6  370.78  5052.3  373.18  5080.8  370.69
  5101.7  370.07  5104.7  369.48  5105.5  368.68  5113.1  368.68  5114.0  369.48
  5115.9  370.11  5137.6  370.29  5186.1  372.96  5265.0  374.65  5534.8  373.45
  5798.0  374.83  5879.0  374.95  5909.4  374.42  6030.9  376.61  6325.2  378.05
#Mann=4,-1,0
  4602.8     0.1       0  5104.7    0.07       0  5114.0     0.1       0
  5186.1    0.05       0
Bank Sta=5104.7,5114
Exp/Cntr=0.3,0.1

Type RM Length L Ch R = 1,16588,70,70,70
BEGIN DESCRIPTION:
Mapping XS 8bb791d7
END DESCRIPTION:
XS GIS Cut Line= 5
      2053954.44     13423275.32      2054148.11     13423084.80
      2054475.80     13422741.92      2054464.83     13422657.29
      2054329.52     13421689.30
#Sta/Elev= 30
  4606.0  390.58  4741.0  387.28  4818.7  383.14  4877.7  381.04  4932.1  376.74
  4967.3  376.99  5005.1  370.21  5005.9  369.41  5013.5  369.41  5014.4  370.21
  5016.7  372.75  5023.9  373.15  5030.8  375.29  5038.0  375.41  5045.0  376.55
  5161.8  375.21  5243.1  374.71  5299.7  375.35  5449.7  373.44  5550.7  373.91
  5591.1  373.23  5712.2  374.52  5830.9  374.92  5934.4  374.28  6005.1  375.72
  6106.0  376.62  6126.8  377.57  6166.6  376.55  6207.0  377.26  6414.7  378.09
#Mann=4,-1,0
  4606.0     0.1       0  5005.1    0.07       0  5014.4     0.1       0
  5161.8    0.05       0
Bank Sta=5005.1,5014.4
Exp/Cntr=0.3,0.1

Type RM Length L Ch R = 1,16518,393,393,393
BEGIN DESCRIPTION:
Mapping XS b709b775
END DESCRIPTION:
XS GIS Cut Line= 4
      2053993.42     13423303.72      2054299.00     13423017.24
      2054522.96     13422772.44      2054397.13     13421739.74
#Sta/Elev= 30
  4591.8  390.19  4613.0  390.05  4705.0  387.53  4854.0  380.62  4903.3  377.23
  4952.7  375.60  4974.2  373.51  4988.3  371.35  4990.5  369.29  4991.4  368.49
  4999.0  368.49  4999.8  369.29  5002.5  369.35  5008.7  371.06  5016.3  370.84
  5023.7  372.27  5030.5  371.63  5037.9  372.74  5052.1  373.34  5157.7  373.59
  5335.1  374.49  5501.1  372.87  5561.5  373.49  5601.8  372.97  5752.9  374.33
  5883.9  374.71  5924.2  374.16  6145.8  377.03  6176.0  376.33  6382.8  377.89
#Mann=5,-1,0
  4591.8    0.05       0  4613.0     0.1       0  4990.5    0.07       0
  4999.8     0.1       0  5157.7    0.05       0
Bank Sta=4990.5,4999.8
Exp/Cntr=0.3,0.1

Type RM Length L Ch R = 1,16125,492,492,492
BEGIN DESCRIPTION:
UNT 059 in RCW 15.0
END DESCRIPTION:
XS GIS Cut Line= 3
      2054440.51     13423681.63      2054625.00     13423125.00
      2054562.14     13421888.20
#Sta/Elev= 30
  4448.2  385.66  4578.1  382.81  4623.7  381.82  4696.5  378.55  4955.4  371.91
  4971.4  371.01  4987.8  368.88  4988.7  368.08  4996.3  368.08  4997.2  368.88
  5013.5  370.67  5024.1  372.40  5032.0  372.75  5144.8  372.27  5174.8  372.96
  5240.0  371.99  5335.1  373.65  5415.1  373.64  5495.2  372.38  5528.7  372.34
  5635.4  373.47  5715.5  372.97  5805.6  374.05  5875.7  373.85  5945.8  374.34
  5985.8  375.14  6065.9  375.15  6126.0  376.07  6206.1  375.69  6273.0  376.56
#Mann=5,-1,0
  4448.2    0.05       0  4578.1     0.1       0  4987.8    0.07       0
  4997.2     0.1       0  5240.0    0.05       0
Bank Sta=4987.8,4997.2
Exp/Cntr=0.3,0.1

Type RM Length L Ch R = 1,15633,470,470,470
BEGIN DESCRIPTION:
UNT 059 in RCW 14.0
END DESCRIPTION:
XS GIS Cut Line= 3
      2054825.00     13424074.99      2054975.00     13423275.00
      2054689.83     13421932.38
#Sta/Elev= 30
  4213.2  400.66  4218.2  400.36  4239.5  398.69  4318.0  396.11  4349.7  395.11
  4417.8  390.13  4454.8  387.74  4565.1  382.93  4681.2  378.52  4762.6  376.48
  4915.2  370.40  4966.1  371.36  4996.1  367.98  4997.0  367.18  5004.6  367.18
  5005.5  367.98  5006.8  368.88  5024.6  370.98  5101.6  372.06  5180.5  371.21
  5313.4  372.20  5339.5  371.20  5344.6  371.87  5374.9  370.20  5405.4  370.22
  5433.6  371.93  5456.5  372.21  5632.1  372.41  5671.2  371.64  6399.7  375.67
#Mann=7,-1,0
  4213.2     0.1       0  4218.2    0.08       0  4318.0    0.05       0
  4417.8     0.1       0  4996.1    0.07       0  5005.5     0.1       0
  5374.9    0.05       0
Bank Sta=4996.1,5005.5
Exp/Cntr=0.3,0.1

Type RM Length L Ch R = 1,15163,67,67,67
BEGIN DESCRIPTION:
Mapping XS 563f4eba
END DESCRIPTION:
XS GIS Cut Line= 6
      2055059.46     13424025.33      2055319.87     13423504.51
      2055351.12     13423330.03      2055299.03     13423244.09
      2055111.53     13423059.20      2054864.40     13422159.11
#Sta/Elev= 30
  4211.2  394.82  4231.6  392.96  4245.1  392.73  4262.6  391.48  4350.5  388.34
  4371.2  387.48  4527.8  381.15  4678.8  376.30  4781.8  371.25  4928.4  368.60
  4973.4  369.06  4995.8  367.69  5012.5  367.60  5013.4  366.80  5021.0  366.80
  5021.9  367.60  5090.2  368.41  5111.4  369.21  5168.0  369.34  5245.8  370.82
  5295.3  370.42  5344.9  371.08  5372.7  370.67  5456.7  371.13  5735.6  371.85
  5794.4  372.48  5849.7  371.66  5932.6  372.39  5982.2  371.76  6270.6  373.59
#Mann=7,-1,0
  4211.2    0.08       0  4262.6    0.05       0  4350.5    0.08       0
  4371.2     0.1       0  5012.5    0.07       0  5021.9     0.1       0
  5456.7    0.05       0
Bank Sta=5012.5,5021.9
Exp/Cntr=0.3,0.1

Type RM Length L Ch R = 1,15096,388,388,388
BEGIN DESCRIPTION:
UNT 059 in RCW 13.0
END DESCRIPTION:
XS GIS Cut Line= 6
      2055082.89     13424046.17      2055408.41     13423486.28
      2055418.83     13423340.45      2055361.53     13423199.82
      2055192.26     13423020.13      2054898.00     13421965.47
#Sta/Elev= 30
  4123.5  394.88  4195.7  390.87  4199.4  390.75  4235.9  388.72  4311.4  386.22
  4380.8  383.05  4594.3  375.77  4680.3  371.50  4888.0  367.76  4888.9  366.96
  4896.6  366.96  4897.5  367.76  4945.5  369.31  4977.2  368.13  5017.6  367.85
  5047.1  368.57  5069.1  368.11  5105.4  369.34  5126.8  368.58  5190.3  370.32
  5226.0  369.50  5296.3  370.36  5390.2  369.97  5653.6  372.51  5766.8  371.25
  5871.6  372.33  5913.2  371.49  6120.8  373.07  6292.0  373.07  6411.0  374.72
#Mann=7,-1,0
  4123.5    0.08       0  4195.7     0.1       0  4199.4    0.08       0
  4311.4     0.1       0  4888.0    0.07       0  4897.5     0.1       0
  5390.2    0.05       0
Bank Sta=4888,4897.5
Exp/Cntr=0.3,0.1

Type RM Length L Ch R = 1,14708,978,978,978
BEGIN DESCRIPTION:
UNT 059 in RCW 12.0
END DESCRIPTION:
XS GIS Cut Line= 4
      2055074.97     13424075.02      2055693.13     13423480.20
      2055949.21     13422681.59      2054815.18     13421458.84
#Sta/Elev= 30
  3910.0  396.22  3969.2  393.27  4043.9  389.53  4181.7  383.58  4235.3  381.46
  4362.7  378.06  4426.2  375.46  4532.5  373.25  4596.0  371.00  4631.5  370.67
  4702.0  368.00  4827.1  367.95  4947.1  368.96  4987.7  367.76  5049.7  368.08
  5277.4  367.69  5278.3  366.89  5286.0  366.89  5286.9  367.69  5342.3  368.09
  5474.9  369.07  5512.3  368.01  5562.6  367.73  5593.7  367.84  5611.6  367.80
  5698.9  367.72  5734.6  369.22  5833.7  370.30  6619.0  373.42  7274.2  378.42
#Mann=12,-1,0
  3910.0    0.08       0  3969.2     0.1       0  4043.9    0.08       0
  4181.7     0.1       0  4947.1    0.07       0  5049.7    0.05       0
  5277.4    0.07       0  5286.9    0.05       0  5342.3     0.1       0
  5562.6    0.05       0  5593.7     0.1       0  5611.6    0.05       0
Bank Sta=5277.4,5286.9
Exp/Cntr=0.3,0.1

Type RM Length L Ch R = 1,13730,95,95,95
BEGIN DESCRIPTION:
UNT 059 in RCW 11.0
END DESCRIPTION:
XS GIS Cut Line= 5
      2055115.89     13424250.15      2055662.75     13423791.84
      2056761.71     13423541.84      2056386.71     13422364.75
      2057308.41     13421109.78
#Sta/Elev= 30
  3039.6  399.43  3444.5  384.92  3559.5  381.51  3592.5  380.06  3852.2  374.26
  5075.1  375.19  5197.5  374.83  5344.7  374.72  5511.2  372.49  5639.9  374.33
  5678.1  371.70  5705.0  374.51  5710.3  371.88  5742.5  371.81  5774.7  374.45
  5780.0  372.09  5825.0  371.52  5929.6  371.36  5935.0  371.78  5941.0  369.35
  6034.2  371.57  6118.3  371.17  6156.8  374.82  6221.6  371.74  6353.9  369.48
  6408.8  366.50  6409.8  365.70  6418.6  366.50  6537.1  372.36  7672.6  374.78
#Mann=17,-1,0
  3039.6     0.1       0  3444.5    0.08       0  3559.5    0.05       0
  3592.5     0.1       0  5075.1    0.05       0  5197.5     0.1       0
  5344.7    0.05       0  5511.2     0.1       0  5639.9    0.05       0
  5825.0     0.1       0  5929.6    0.05       0  5935.0    0.07       0
  6034.2     0.1       0  6221.6    0.05       0  6353.9     0.1       0
  6408.8    0.07       0  6418.6     0.1       0
Bank Sta=6408.8,6418.6
Exp/Cntr=0.3,0.1

Type RM Length L Ch R = 1,13635,400,400,400
BEGIN DESCRIPTION:
UNT 059 in RCW 10.0
END DESCRIPTION:
XS GIS Cut Line= 6
      2055176.64     13424313.54      2055733.93     13423849.13
      2056860.67     13423567.01      2056500.42     13422351.73
      2057190.53     13421587.84      2057429.25     13421175.51
#Sta/Elev= 30
  2971.7  394.04  3033.9  392.95  3161.5  396.12  3352.8  385.93  3470.4  381.87
  3537.9  378.93  3791.0  370.62  4471.0  366.74  4599.8  367.61  4677.0  366.26
  4682.2  367.57  4759.4  366.11  4770.3  367.20  4817.0  365.65  4817.9  364.85
  4826.8  365.65  5197.1  366.94  5356.3  367.51  5508.7  368.24  5669.4  369.08
  5716.4  369.41  6148.7  372.17  6247.4  371.39  6320.8  366.70  6346.7  366.19
  6381.9  370.21  6410.3  371.43  6538.0  372.14  7175.4  371.05  7632.1  373.80
#Mann=11,-1,0
  2971.7     0.1       0  3470.4    0.05       0  3537.9     0.1       0
  4817.0    0.07       0  4826.8     0.1       0  5197.1    0.05       0
  5356.3     0.1       0  5508.7    0.05       0  5669.4     0.1       0
  5716.4    0.05       0  6320.8     0.1       0
Bank Sta=4817,4826.8
Exp/Cntr=0.3,0.1

Type RM Length L Ch R = 1,13235,686,686,686
BEGIN DESCRIPTION:
Mapping XS 98c47a65
END DESCRIPTION:
XS GIS Cut Line= 4
      2057039.14     13424142.66      2057167.18     13423528.54
      2057425.83     13422436.42      2057520.88     13421189.59
#Sta/Elev= 30
  4258.7  366.74  4481.0  365.44  4602.2  363.11  4621.2  361.20  4634.3  360.21
  4664.9  364.35  4910.2  363.45  4951.3  361.58  5002.7  357.17  5057.6  360.17
  5126.0  359.47  5151.5  362.11  5177.4  363.79  5249.9  362.84  5300.7  358.88
  5321.3  358.53  5336.9  356.23  5337.9  355.43  5346.8  356.23  5371.6  360.56
  5382.9  360.97  5424.1  360.90  5475.4  363.20  5670.7  366.61  5886.5  363.50
  6070.0  367.90  6571.4  370.05  6701.8  369.24  6723.9  370.49  7258.8  373.63
#Mann=6,-1,0
  4258.7    0.05       0  4621.2     0.1       0  5057.6    0.07       0
  5151.5     0.1       0  5336.9    0.07       0  5346.8     0.1       0
Bank Sta=5336.9,5346.8
Exp/Cntr=0.3,0.1

Type RM Length L Ch R = 1,12549,496,496,496
BEGIN DESCRIPTION:
Mapping XS 2ca16296
END DESCRIPTION:
XS GIS Cut Line= 3
      2057215.71     13423875.15      2057531.67     13423375.17
      2057614.83     13422578.25
#Sta/Elev= 30
  4263.1  364.48  4283.6  364.21  4349.0  362.48  4364.3  360.33  4393.4  359.25
  4416.0  360.00  4421.9  358.96  4437.2  361.06  4443.1  360.08  4567.8  363.58
  4683.1  363.43  4813.7  360.99  4842.9  362.52  4945.2  362.58  5000.1  355.12
  5000.9  354.32  5011.0  355.12  5030.9  355.14  5055.8  357.56  5099.8  359.44
  5166.4  362.61  5206.6  360.83  5222.8  357.90  5236.8  357.29  5249.4  358.34
  5277.0  360.30  5357.4  359.04  5377.5  361.23  5419.7  362.87  5655.8  365.53
#Mann=6,-1,0
  4263.1    0.05       0  4283.6     0.1       0  5000.1    0.07       0
  5011.0     0.1       0  5099.8    0.12       0  5249.4     0.1       0
Bank Sta=5000.1,5011
Exp/Cntr=0.3,0.1

Type RM Length L Ch R = 1,12053,429,429,429
BEGIN DESCRIPTION:
Mapping XS 5c7f0abb
END DESCRIPTION:
XS GIS Cut Line= 4
      2057226.10     13424027.97      2057594.17     13423420.31
      2058021.26     13422944.61      2058305.94     13422757.14
#Sta/Elev= 30
  3931.1  365.51  4089.1  363.81  4203.2  362.12  4245.9  358.69  4261.4  358.96
  4304.1  362.53  4507.5  363.28  4667.0  361.13  4723.8  361.96  4830.0  360.88
  4844.2  361.72  4865.1  359.10  4872.6  359.14  4893.5  357.03  4978.8  355.13
  4994.2  352.96  4995.0  352.16  5004.3  352.16  5005.1  352.96  5021.4  353.89
  5028.1  356.02  5035.6  355.93  5042.3  357.25  5135.7  361.21  5247.9  360.46
  5311.3  356.59  5347.5  359.76  5455.9  360.53  5507.1  362.19  5621.7  362.86
#Mann=5,-1,0
  3931.1    0.05       0  4089.1     0.1       0  4994.2    0.07       0
  5005.1     0.1       0  5135.7     0.1       0
Bank Sta=4994.2,5005.1
Exp/Cntr=0.3,0.1

Type RM Length L Ch R = 1,11624,742,742,742
BEGIN DESCRIPTION:
Mapping XS caec6862
END DESCRIPTION:
XS GIS Cut Line= 3
      2057476.13     13423993.21      2057740.01     13423427.25
      2058340.37     13422854.65
#Sta/Elev= 30
  3768.1  364.65  3912.6  363.13  3968.4  362.50  4065.4  358.00  4141.3  357.91
  4156.9  358.31  4163.3  360.01  4185.4  362.09  4276.7  362.85  4496.5  360.90
  4539.0  357.86  4581.5  359.80  4617.0  358.39  4623.9  359.25  4631.2  358.22
  4638.1  359.47  4645.3  358.07  4666.4  359.32  4727.2  355.15  4744.4  354.20
  4765.5  356.27  4800.7  357.08  4885.9  356.94  4928.1  356.74  4984.4  354.56
  4993.4  353.63  4994.1  352.83  5004.3  353.63  5076.6  358.75  5222.2  361.01
#Mann=7,-1,0
  3768.1    0.05       0  3912.6     0.1       0  4727.2    0.12       0
  4885.9    0.07       0  4984.4     0.1       0  4993.4    0.07       0
  5004.3     0.1       0
Bank Sta=4993.4,5004.3
Exp/Cntr=0.3,0.1

Type RM Length L Ch R = 1,10882,174,174,174
BEGIN DESCRIPTION:
Mapping XS fa8e5524
END DESCRIPTION:
XS GIS Cut Line= 4
      2057726.12     13424104.34      2058055.98     13423805.73
      2058184.45     13423312.67      2058406.66     13422823.11
#Sta/Elev= 30
  4271.4  364.62  4666.5  361.45  4709.1  363.89  4732.4  363.79  4767.8  362.93
  4799.8  359.70  4813.2  356.48  4848.8  353.06  4889.3  351.41  4913.4  351.81
  4929.8  354.71  4934.9  353.05  4965.1  354.06  4990.7  348.66  4991.4  347.86
  5001.6  348.66  5016.8  351.85  5046.1  354.31  5099.5  353.44  5132.3  354.41
  5151.1  357.14  5182.1  359.06  5234.0  356.49  5344.1  360.77  5412.1  357.23
  5458.2  356.75  5481.3  358.03  5519.8  357.13  5653.8  360.33  5763.5  361.07
#Mann=4,-1,0
  4271.4    0.05       0  4813.2     0.1       0  4990.7    0.07       0
  5001.6     0.1       0
Bank Sta=4990.7,5001.6
Exp/Cntr=0.3,0.1

Type RM Length L Ch R = 1,10708,415,415,415
BEGIN DESCRIPTION:
UNT 059 in RCW 9.0
END DESCRIPTION:
XS GIS Cut Line= 3
      2058139.30     13424055.76      2058378.57     13423263.84
      2058496.94     13422854.38
#Sta/Elev= 30
  4492.4  363.11  4505.0  363.00  4570.4  362.67  4681.2  361.99  4796.1  359.56
  4907.8  358.83  4940.7  356.77  4963.3  354.05  4978.9  351.20  4984.2  348.54
  4999.6  346.46  5000.4  345.66  5009.8  345.66  5010.5  346.46  5011.9  348.50
  5044.8  355.99  5057.3  358.54  5067.7  358.84  5148.9  359.10  5193.1  357.86
  5253.0  358.85  5308.0  358.92  5329.5  357.78  5357.9  357.41  5401.9  355.22
  5463.9  359.46  5536.4  358.31  5575.2  359.01  5620.3  358.73  5745.9  361.02
#Mann=5,-1,0
  4492.4    0.05       0  4505.0     0.1       0  4570.4    0.05       0
  4999.6    0.03       0  5010.5     0.1       0
Bank Sta=4999.6,5010.5
Exp/Cntr=0.3,0.1

Type RM Length L Ch R = 1,10293,681,681,681
BEGIN DESCRIPTION:
Mapping XS dfdd4414
END DESCRIPTION:
XS GIS Cut Line= 3
      2058274.71     13424045.35      2058517.78     13423573.09
      2058639.32     13422913.34
#Sta/Elev= 30
  4374.7  361.41  4402.6  361.27  4532.6  360.81  4656.3  357.91  4716.1  358.59
  4768.7  354.63  4822.1  352.45  4826.9  353.80  4843.5  353.19  4849.1  353.84
  4905.9  353.26  4924.2  351.35  4976.7  352.39  5000.1  347.69  5000.9  346.89
  5010.3  346.89  5011.0  347.69  5015.8  348.58  5024.7  352.70  5029.7  351.85
  5036.1  354.97  5046.3  357.71  5076.8  359.49  5140.9  358.81  5199.0  352.78
  5299.9  357.48  5416.1  355.74  5442.8  357.95  5483.5  357.66  5576.7  360.32
#Mann=5,-1,0
  4374.7     0.1       0  4402.6    0.05       0  4822.1     0.1       0
  5000.1    0.07       0  5011.0     0.1       0
Bank Sta=5000.1,5011
Exp/Cntr=0.3,0.1

Type RM Length L Ch R = 1,9612,1433,1433,1433
BEGIN DESCRIPTION:
UNT 059 in RCW 8.0
END DESCRIPTION:
XS GIS Cut Line= 3
      2058546.98     13424567.63      2058709.03     13423796.53
      2058781.35     13422900.99
#Sta/Elev= 30
  4251.1  362.32  4285.6  362.52  4606.2  361.39  4724.7  356.74  4744.3  355.72
  4755.8  352.60  4774.9  352.94  4805.7  350.11  4887.3  351.53  4918.0  353.99
  4989.5  349.75  4992.6  348.57  5004.5  345.18  5005.3  344.38  5015.4  345.18
  5042.3  347.31  5053.4  353.21  5060.6  355.22  5090.7  358.56  5112.9  359.20
  5321.5  359.09  5371.7  353.66  5431.8  358.95  5492.0  359.40  5632.5  350.81
  5652.6  352.42  5712.8  353.12  5783.0  358.69  5873.3  359.58  5937.5  357.64
#Mann=7,-1,0
  4251.1     0.1       0  4285.6    0.05       0  4724.7     0.1       0
  4992.6    0.12       0  5004.5    0.07       0  5015.4    0.12       0
  5112.9     0.1       0
Bank Sta=5004.5,5015.4
Exp/Cntr=0.3,0.1

Type RM Length L Ch R = 1,8179,543,543,543
BEGIN DESCRIPTION:
Mapping XS 2013079d
END DESCRIPTION:
XS GIS Cut Line= 4
      2059156.67     13424371.74      2059208.76     13423805.73
      2058847.64     13423392.53      2058903.20     13422691.19
#Sta/Elev= 30
  4009.2  356.34  4277.1  356.16  4307.2  353.11  4357.4  351.64  4372.7  349.04
  4407.6  348.68  4462.4  342.24  4463.2  341.44  4473.4  342.24  4488.0  345.57
  4528.1  349.94  4616.5  349.19  4764.6  351.17  4899.4  350.37  4970.6  346.80
  4991.5  343.56  5005.7  343.41  5013.3  343.71  5019.9  347.96  5027.5  348.45
  5034.2  351.45  5056.0  356.65  5124.6  358.22  5304.4  349.51  5414.8  356.09
  5495.0  352.10  5595.4  350.95  5666.7  354.85  5715.7  353.58  5829.9  354.88
#Mann=3,-1,0
  4009.2     0.1       0  4462.4    0.07       0  4473.4     0.1       0
Bank Sta=4462.4,4473.4
Exp/Cntr=0.3,0.1

Type RM Length L Ch R = 1,7636,444,444,444
BEGIN DESCRIPTION:
Mapping XS dbd209d6
END DESCRIPTION:
XS GIS Cut Line= 2
      2059236.54     13424441.10      2059298.95     13423158.22
#Sta/Elev= 30
  4122.4  355.70  4193.6  356.10  4368.8  355.08  4458.9  355.88  4497.0  353.97
  4569.0  351.92  4604.7  352.25  4609.7  351.21  4649.1  348.99  4699.2  349.10
  4749.2  347.29  4799.3  349.28  4849.4  354.31  4869.4  354.34  4919.4  347.68
  4969.5  346.23  4989.5  341.85  4994.0  338.99  4994.7  338.19  5004.4  338.19
  5005.1  338.99  5015.7  345.04  5020.7  344.70  5049.6  355.15  5069.6  357.48
  5109.7  357.55  5149.7  355.10  5209.8  354.61  5239.8  352.77  5406.8  357.92
#Mann=4,-1,0
  4122.4    0.05       0  4497.0     0.1       0  4994.0    0.07       0
  5005.1     0.1       0
Bank Sta=4994,5005.1
Exp/Cntr=0.3,0.1

Type RM Length L Ch R = 1,7192,83,83,83
BEGIN DESCRIPTION:
Mapping XS ffb7f35b
END DESCRIPTION:
XS GIS Cut Line= 5
      2059326.81     13424423.75      2059371.95     13423649.48
      2059500.42     13423569.61      2059587.23     13423611.28
      2060125.46     13423177.22
#Sta/Elev= 30
  4016.7  355.04  4265.9  355.29  4399.6  350.77  4516.3  348.60  4566.4  346.19
  4676.6  353.30  4766.7  346.68  4863.9  346.20  4900.5  343.27  4959.7  343.47
  4998.6  340.49  4999.3  339.69  5009.7  340.49  5038.4  349.47  5042.7  348.34
  5057.0  351.88  5063.5  350.78  5071.4  351.94  5077.9  350.06  5085.8  350.59
  5092.2  348.98  5100.2  349.92  5106.6  348.88  5121.0  351.18  5135.4  350.76
  5156.2  347.60  5199.4  349.92  5284.2  358.32  5420.4  359.65  5731.3  359.71
#Mann=5,-1,0
  4016.7    0.05       0  4399.6     0.1       0  4998.6    0.07       0
  5009.7     0.1       0  5420.4    0.05       0
Bank Sta=4998.6,5009.7
Exp/Cntr=0.3,0.1

Type RM Length L Ch R = 1,7109,368,368,368
BEGIN DESCRIPTION:
Mapping XS f253418c
END DESCRIPTION:
XS GIS Cut Line= 4
      2059340.70     13424409.88      2059427.51     13423666.84
      2059632.37     13423670.31      2060194.90     13423194.59
#Sta/Elev= 30
  4148.6  355.16  4385.1  355.07  4489.0  353.84  4529.1  351.52  4616.6  347.80
  4797.9  348.82  4868.3  345.77  4934.2  346.11  4964.2  345.05  5008.7  340.71
  5009.4  339.91  5019.8  340.71  5086.3  342.55  5100.4  341.32  5149.7  344.47
  5170.5  346.63  5178.3  348.69  5184.8  346.95  5192.6  348.88  5199.1  347.59
  5206.9  348.37  5213.4  346.84  5221.2  348.34  5227.7  347.64  5256.3  350.22
  5270.6  349.65  5277.1  351.38  5340.8  355.96  5493.4  359.35  5838.3  359.94
#Mann=5,-1,0
  4148.6    0.05       0  4529.1     0.1       0  5008.7    0.07       0
  5019.8     0.1       0  5493.4    0.05       0
Bank Sta=5008.7,5019.8
Exp/Cntr=0.3,0.1

Type RM Length L Ch R = 1,6741,336,336,336
BEGIN DESCRIPTION:
Mapping XS 919ead23
END DESCRIPTION:
XS GIS Cut Line= 2
      2059515.16     13424210.27      2060304.05     13423178.63
#Sta/Elev= 30
  4502.7  353.76  4534.5  353.27  4671.0  355.04  4820.6  354.43  4891.3  350.71
  4955.7  345.66  4976.5  342.77  4991.0  339.80  4993.7  338.51  4994.4  337.71
  5004.1  337.71  5004.8  338.51  5026.4  343.39  5049.1  346.63  5134.4  352.78
  5184.2  352.53  5190.5  350.89  5198.8  351.40  5205.0  350.31  5219.6  352.44
  5234.1  351.62  5240.4  352.43  5248.6  351.31  5254.9  352.66  5277.2  353.64
  5319.3  358.40  5340.2  357.18  5385.1  359.75  5769.7  359.81  5801.4  359.98
#Mann=5,-1,0
  4502.7     0.1       0  4993.7    0.07       0  5004.8     0.1       0
  5385.1    0.05       0  5769.7     0.1       0
Bank Sta=4993.7,5004.8
Exp/Cntr=0.3,0.1

Type RM Length L Ch R = 1,6405,428,428,428
BEGIN DESCRIPTION:
Mapping XS fd501f1b
END DESCRIPTION:
XS GIS Cut Line= 2
      2059528.21     13424479.33      2060504.78     13423485.40
#Sta/Elev= 30
  4124.1  354.86  4216.8  353.59  4259.2  351.56  4294.6  346.30  4308.8  346.58
  4344.1  351.99  4400.6  354.04  4683.5  352.30  4789.5  346.12  4931.0  344.75
  4973.4  341.01  4980.5  337.30  5001.7  338.01  5010.3  336.51  5011.0  335.71
  5021.4  336.51  5023.0  339.28  5030.0  338.75  5037.1  341.00  5051.3  341.32
  5093.7  349.44  5114.8  349.93  5122.0  352.87  5129.0  351.98  5136.1  354.33
  5143.1  354.11  5150.3  356.29  5157.3  355.72  5218.4  359.55  5517.5  359.80
#Mann=4,-1,0
  4124.1     0.1       0  5010.3    0.07       0  5021.4     0.1       0
  5218.4    0.05       0
Bank Sta=5010.3,5021.4
Exp/Cntr=0.3,0.1

Type RM Length L Ch R = 1,5977,737,737,737
BEGIN DESCRIPTION:
Mapping XS 15a67380
END DESCRIPTION:
XS GIS Cut Line= 2
      2059419.73     13424613.87      2060591.61     13424058.31
#Sta/Elev= 30
  4002.8  354.13  4135.9  355.14  4223.2  354.40  4245.9  353.05  4291.4  346.21
  4329.6  343.80  4410.6  351.99  4450.6  350.39  4456.1  351.92  4473.3  351.10
  4478.8  352.31  4529.9  354.95  4660.8  344.56  4711.8  341.99  4950.2  342.64
  4967.4  340.92  4973.0  341.51  4990.2  338.23  4999.1  337.92  4999.8  337.12
  5010.2  337.92  5012.9  339.15  5018.4  339.02  5035.6  346.26  5041.2  345.74
  5058.4  352.09  5063.5  350.87  5093.2  357.54  5115.3  360.20  5299.7  360.15
#Mann=5,-1,0
  4002.8    0.05       0  4135.9     0.1       0  4999.1    0.07       0
  5010.2     0.1       0  5063.5    0.05       0
Bank Sta=4999.1,5010.2
Exp/Cntr=0.3,0.1

Type RM Length L Ch R = 1,5240,448,448,448
BEGIN DESCRIPTION:
UNT 059 in RCW 6.0
END DESCRIPTION:
XS GIS Cut Line= 3
      2059425.04     13425024.99      2060225.00     13424725.00
      2060425.01     13424374.98
#Sta/Elev= 30
  4172.8  357.57  4303.6  354.99  4353.4  351.78  4358.8  352.65  4383.7  348.21
  4389.0  349.83  4395.4  348.61  4414.0  346.42  4419.3  347.51  4444.2  347.53
  4493.2  346.14  4584.8  353.35  4664.0  352.01  4738.8  353.46  4802.9  352.95
  4888.3  349.66  4926.6  342.99  4956.9  339.98  4973.8  336.57  4976.2  334.61
  4976.9  333.81  4987.4  334.61  5012.0  335.93  5017.4  337.80  5030.0  338.04
  5062.4  342.38  5180.5  346.30  5261.1  353.29  5309.0  355.50  5430.3  358.50
#Mann=5,-1,0
  4172.8    0.05       0  4395.4     0.1       0  4976.2    0.07       0
  4987.4     0.1       0  5309.0    0.05       0
Bank Sta=4976.2,4987.4
Exp/Cntr=0.3,0.1

Type RM Length L Ch R = 1,4792,800,800,800
BEGIN DESCRIPTION:
UNT 059 in RCW 5.0
END DESCRIPTION:
XS GIS Cut Line= 3
      2060301.29     13425347.22      2060475.00     13425025.00
      2060833.88     13424458.82
#Sta/Elev= 30
  4636.7  350.23  4684.7  349.89  4767.2  350.79  4832.4  351.77  4907.1  351.96
  4929.0  351.69  4945.2  350.65  4950.9  349.82  4972.8  343.09  4980.0  339.01
  4994.3  334.41  4995.1  333.61  5004.8  333.61  5005.5  334.41  5010.4  336.32
  5016.3  337.48  5031.6  338.88  5119.7  339.59  5156.1  340.56  5219.7  340.11
  5240.9  341.64  5271.4  345.77  5307.8  348.09  5350.2  351.74  5386.6  353.14
  5401.9  352.30  5429.0  352.63  5465.3  354.84  5517.1  356.48  5673.1  358.72
#Mann=5,-1,0
  4636.7    0.05       0  4767.2     0.1       0  4994.3    0.07       0
  5005.5     0.1       0  5465.3    0.05       0
Bank Sta=4994.3,5005.5
Exp/Cntr=0.3,0.1
