--- San Miguel Creek.prj (project) ---

Proj Title=San Miguel Creek Base Level Engineering
Current Plan=p01
Default Exp/Contr=0.3,0.1
English Units
Geom File=g01
Flow File=f01
Plan File=p01
Y Axis Title=Elevation
X Axis Title(PF)=Main Channel Distance
X Axis Title(XS)=Station
BEGIN DESCRIPTION:
San Miguel Creek
END DESCRIPTION:
DSS Export Rating Curves= 0
DSS Export Rating Curve Sorted= 0
DSS Export Volume Flow Curves= 0
DXF OffsetX= 0
DXF OffsetY= 0
DXF ScaleX= 1
DXF ScaleY= 10

--- San Miguel Creek.p01 (plan) ---

Plan Title=Multiple Run
Short Identifier=Multiple
Geom File=g01
Flow File=f01
Subcritical Flow
K Sum by GR= 0
Std Step Tol= 0.01
Critical Tol= 0.01
Num of Std Step Trials= 20
Max Error Tol= 0.3
Flow Tol Ratio= 0.001
Split Flow NTrial= 30
Split Flow Tol= 0.02
Split Flow Ratio= 0.02
Log Output Level= 0
Friction Slope Method= 1
Unsteady Friction Slope Method= 2
Unsteady Bridges Friction Slope Method= 1
Parabolic Critical Depth
Global Vel Dist=  1 , 1 , 1
Global Log Level= 0
CheckData=True
Encroach Param= -1, 0, 0, 0
BEGIN DESCRIPTION:
Multiple Run
END DESCRIPTION:

--- San Miguel Creek.f01 (steady flow) ---

Flow Title=Multiple
Program Version=5.07
BEGIN FILE DESCRIPTION:
Gage 08206700 analysis results and adjusted with 1996-4307 regression equation flows, see spreadsheet for details.
END FILE DESCRIPTION:
Number of Profiles= 7
Profile Names=10-year,25-year,50-year,1pct_min,100-year,1pct_plu,500-year
River Rch & RM=San Miguel Creek,Reach-1         ,412100
    4350    7660   11000    8050   15700   30600   35800
River Rch & RM=San Miguel Creek,Reach-1         ,410686
    5870   10300   14800    9860   19200   37500   35800
River Rch & RM=San Miguel Creek,Reach-1         ,296851
    7050   12300   17600   12000   23400   45600   45500
River Rch & RM=San Miguel Creek,Reach-1         ,292935
    8070   13900   19800   13100   25500   49600   46000
River Rch & RM=San Miguel Creek,Reach-1         ,239193
    8890   15100   21100   13700   26800   52200   46500
River Rch & RM=San Miguel Creek,Reach-1         ,191995
   10000   16600   22800   14500   28300   55200   46800
River Rch & RM=San Miguel Creek,Reach-1         ,113058
   12200   19200   25200   16100   31300   61000   48200
River Rch & RM=San Miguel Creek,Reach-1         ,68755
   12700   20300   27100   16900   32900   64200   48500
Boundary for River Rch & Prof#=San Miguel Creek,Reach-1         , 1
Up Type= 0
Dn Type= 3
Dn Slope=0.0001
Boundary for River Rch & Prof#=San Miguel Creek,Reach-1         , 2
Up Type= 0
Dn Type= 3
Dn Slope=0.0001
Boundary for River Rch & Prof#=San Miguel Creek,Reach-1         , 3
Up Type= 0
Dn Type= 3
Dn Slope=0.0001
Boundary for River Rch & Prof#=San Miguel Creek,Reach-1         , 4
Up Type= 0
Dn Type= 3
Dn Slope=0.0001
Boundary for River Rch & Prof#=San Miguel Creek,Reach-1         , 5
Up Type= 0
Dn Type= 3
Dn Slope=0.0001
Boundary for River Rch & Prof#=San Miguel Creek,Reach-1         , 6
Up Type= 0
Dn Type= 3
Dn Slope=0.0001
Boundary for River Rch & Prof#=San Miguel Creek,Reach-1         , 7
Up Type= 0
Dn Type= 3
Dn Slope=0.0001
DSS Import GetInterval= 0
DSS Import GetPeak= 0
DSS Import FillOption= 0

--- San Miguel Creek.g01 (geometry) ---

Geom Title=Existing Conditions
Program Version=5.07

River Reach=San Miguel Creek,Reach-1
Reach XY= 30
       1990930.8     13579164.54       1985830.8     13570444.54
      1986607.83      13553456.7       1982950.8     13541504.54
       1994880.8     13529724.54       1992100.8     13525084.54
       1997980.8     13515004.54      1994990.34     13499573.07
       2009240.8     13458184.54       2018220.8     13453534.54
       2019910.8     13446134.54       2027130.8     13438984.54
       2042690.8     13441394.54       2047810.8     13436604.54
      2058867.62     13434504.47       2060140.8     13430064.54
       2070540.8     13423034.54       2078170.8     13424534.54
       2086530.8     13418344.54       2089890.8     13420574.54
       2098920.8     13413294.54       2099630.8     13407884.54
       2109810.8     13403914.54       2111770.8     13397664.54
       2125210.8     13396624.54       2131890.8     13381204.54
       2139711.1     13375536.34       2142916.4     13377648.97
      2151254.17     13370232.41      2155128.48     13370999.29

Type RM Length L Ch R = 1 ,412100  ,1414,1414,1414
BEGIN DESCRIPTION:
San Miguel Creek 228.0
END DESCRIPTION:
XS GIS Cut Line= 3
      1993700.01       13578700.       1990930.8     13579164.54
      1988569.11      13579796.2
#Sta/Elev= 30
  2192.1  631.52  2737.9   626.1  3341.8  611.84  3521.2  606.61  3735.9  600.66
  3943.1  598.71  4157.9   601.9  4770.8  598.84  4913.4  598.44  4932.4   594.9
  4962.8  593.44  4967.9  591.76    4974  587.07  4980.2  586.66  4987.5  585.66
  5015.6  586.66  5018.8  591.49  5024.1  592.36  5075.9  593.05    5134  596.78
  5277.7  598.75  5524.8  596.54  5655.6  598.62  5841.9  608.03  6046.5  614.29
  6488.9  618.28  6525.1  620.12  7099.6  628.82  7321.7  630.86  7444.7  629.93
#Mann= 8 ,-1 , 0
  2192.1     .05       0  3341.8     .12       0  3521.2     .05       0
  4770.8     .12       0  4980.2     .07       0  5015.6     .12       0
    5134      .1       0  5524.8     .05       0
Bank Sta=4980.2,5015.6
XS Rating Curve= 0 ,0
Exp/Cntr=0.3,0.1

Type RM Length L Ch R = 1 ,410686  ,1244,1244,1244
BEGIN DESCRIPTION:
San Miguel Creek 227.0
END DESCRIPTION:
XS GIS Cut Line= 3
      1994668.59     13577563.61       1990115.5       13578095.
      1987904.73     13579247.41
#Sta/Elev= 30
     416  621.91   772.5  614.44  1376.5  607.71  2540.2  599.76  3397.2   599.9
    4869   595.4  4897.3  594.86  4958.5  597.67  4987.9  592.34  4990.7  585.37
  4998.1  584.37  5026.4  585.37  5030.6  594.14  5055.5  590.26    5071  590.99
  5077.8  593.04  5096.9  596.09  5110.7  595.04  5292.9  601.81  5403.7   608.6
  5497.2  611.96  5589.8  612.52    5638  615.09  5911.3  615.12  6038.2  618.69
    6317  620.53  6587.5   623.7  6678.7  626.53  6935.4  627.69  7493.1  634.73
#Mann= 5 ,-1 , 0
     416     .05       0    4869     .12       0  4990.7     .07       0
  5026.4     .12       0  5077.8     .05       0
Bank Sta=4990.7,5026.4
XS Rating Curve= 0 ,0
Exp/Cntr=0.3,0.1

Type RM Length L Ch R = 1 ,409442  ,115,115,115
BEGIN DESCRIPTION:
San Miguel Creek 226.0
END DESCRIPTION:
XS GIS Cut Line= 6
      1994164.63     13576879.14      1991628.04     13576943.75
      1990218.16     13577038.15      1989555.98     13577085.22
      1989178.22      13577131.9      1987623.05     13578724.77
#Sta/Elev= 30
   385.7  619.91  1599.2  610.45  1910.8  612.21  2137.9  610.87  2206.2  608.36
  2304.7  604.11  2363.5  602.15  2600.1  600.31  2743.6  594.45  2813.6  600.05
  3016.5  597.31  4673.9  594.98  4772.8  595.12  4858.3  596.51  4871.6  594.93
  4923.3  592.71  4953.4  594.37  4970.4  589.11  4978.4  586.13  4978.6  584.09
    4986  583.09  5014.3  584.09  5028.7  594.84  5069.7  599.61  5270.5   610.5
  5614.9  621.27  5809.4  624.98  6223.1  625.84  6622.6   623.6  7606.8  630.02
#Mann= 13 ,-1 , 0
   385.7     .05       0  1910.8     .08       0  2137.9     .05       0
  2206.2      .1       0  2304.7     .08       0  2600.1     .05       0
  4673.9     .07       0  4772.8     .12       0  4871.6     .16       0
  4970.4     .12       0  4978.6     .07       0  5014.3     .12       0
  5069.7     .05       0
Bank Sta=4978.6,5014.3
XS Rating Curve= 0 ,0
Exp/Cntr=0.3,0.1

Type RM Length L Ch R = 1 ,409327  ,1184,1184,1184
BEGIN DESCRIPTION:
Mapping XS 7335b55c
END DESCRIPTION:
XS GIS Cut Line= 5
      1994012.13     13576672.07      1990195.59     13576909.67
      1989542.28     13576973.98      1989096.98     13577011.25
      1987538.28     13578598.69
#Sta/Elev= 30
   519.6   620.9   614.4  621.99  1676.5  609.65  1982.1  613.96  2014.9   615.8
  2122.3  611.79  2197.5  611.54  2242.6  608.43  2496.8  599.88    3009   596.3
  4754.7  593.91  4853.9  593.27    4953  594.44  4969.6  593.72  4974.7  590.81
  4976.9  583.96  4984.3  582.96  5012.6  583.96  5014.8  586.67  5024.9  585.58
  5029.9  586.98  5039.9  594.56  5062.1  596.72  5225.6  606.65  5613.1  618.84
  6228.7  627.15  6288.9  625.38    6646  625.04  7381.4   628.3  7671.6  627.04
#Mann= 8 ,-1 , 0
   519.6     .05       0  4754.7     .07       0  4853.9     .12       0
    4953     .16       0  4976.9     .07       0  5012.6     .16       0
  5062.1      .1       0  5613.1     .05       0
Bank Sta=4976.9,5012.6
XS Rating Curve= 0 ,0
Exp/Cntr=0.3,0.1

Type RM Length L Ch R = 1 ,408143  ,1615,1615,1615
BEGIN DESCRIPTION:
San Miguel Creek 225.0
END DESCRIPTION:
XS GIS Cut Line= 3
      1992106.07     13573881.93      1989260.15     13575876.19
      1987340.24     13578327.66
#Sta/Elev= 30
  1524.9  632.68  1739.6  625.37  1955.4   622.7    2012  620.24  2087.9  621.41
  2116.2  620.53    2131  618.56  2270.9  614.26    2964  608.47  3104.3  608.71
  4159.6  591.68  4884.9  593.03  4966.6  592.96  4973.8  591.75  4988.6  584.67
  4988.7  583.45  4996.1  582.45    5017  582.45  5024.4  583.45  5027.4  591.13
  5051.1   592.2  5085.9   593.2  5165.3  595.03  5560.8  598.41  5576.2  598.54
    5605  601.15  5786.4   607.3  5982.2  608.52  6623.2  624.69  8113.8  622.18
#Mann= 8 ,-1 , 0
  1524.9     .05       0  4884.9     .12       0  4988.7     .07       0
  5024.4     .12       0  5051.1      .1       0  5085.9     .07       0
  5165.3      .1       0  5560.8     .05       0
Bank Sta=4988.7,5024.4
XS Rating Curve= 0 ,0
Exp/Cntr=0.3,0.1

Type RM Length L Ch R = 1 ,406528  ,2039,2039,2039
BEGIN DESCRIPTION:
San Miguel Creek 224.0
END DESCRIPTION:
XS GIS Cut Line= 3
      1991425.44     13572963.45       1988400.8     13575094.54
      1986628.94     13577776.25
#Sta/Elev= 30
    1300     640  1778.9  628.16  1943.9  621.47  2299.3  612.36  3142.3  598.45
  4035.9  589.25    4874  592.43  4911.6  592.57  4979.6  590.04    4983  589.41
  4983.2  578.59  4990.6  577.59  5018.9  578.59  5019.1  582.64  5033.5  587.95
  5059.1  590.28    5153  591.35  5225.2  589.87  5661.7  596.73  5943.1  604.19
  5982.2  603.81  6028.8  606.92  6098.1  608.07  6353.9  609.34  6408.1  608.57
  6495.4  609.77  6570.6  607.18    6852  606.53  7596.6  611.97  8214.2  617.18
#Mann= 6 ,-1 , 0
    1300     .05       0    4874     .12       0  4983.2     .07       0
  5018.9     .12       0  5059.1      .1       0  7596.6     .05       0
Bank Sta=4983.2,5018.9
XS Rating Curve= 0 ,0
Exp/Cntr=0.3,0.1

Type RM Length L Ch R = 1 ,404489  ,1906,1906,1906
BEGIN DESCRIPTION:
San Miguel Creek 223.0
END DESCRIPTION:
XS GIS Cut Line= 3
      1991555.67     13572650.93        1987025.       13574125.
      1983904.45     13575709.68
#Sta/Elev= 30
   256.4   652.3  1061.5  627.16  1255.7  625.81  1351.5  627.01  2016.7  611.64
  2415.5  609.03  2692.6  611.96  2851.9  609.78  3509.2  587.34  4339.7  592.05
  4877.6  590.94  4944.6  587.45  4972.9  587.75  4981.4  586.54    4987  576.33
  4994.4  575.33  5022.7  576.33  5023.6  587.12  5034.9   591.3  5051.8  591.71
  5371.3  592.19  5738.6  595.54  6044.3  590.85  7041.8  601.58  7153.9  602.71
    7266  604.39  7642.5  609.98  8036.7  611.71  8476.2  623.21  8520.7  621.61
#Mann= 8 ,-1 , 0
   256.4     .05       0  4877.6     .12       0    4987     .07       0
  5022.7     .12       0  5051.8     .05       0  7041.8      .1       0
  7153.9     .08       0    7266      .1       0
Bank Sta=4987,5022.7
XS Rating Curve= 0 ,0
Exp/Cntr=0.3,0.1

Type RM Length L Ch R = 1 ,402583  ,1629,1629,1629
BEGIN DESCRIPTION:
San Miguel Creek 222.0
END DESCRIPTION:
XS GIS Cut Line= 3
      1990465.73     13572238.08       1987510.8     13572874.54
      1983261.02      13574739.8
#Sta/Elev= 30
  1977.3   629.3  2366.6  622.68    2625  621.97  3696.4  604.83    4573  599.04
    4666  595.64  4753.4  592.44  4880.6  587.42  4957.3  587.56  4967.6  585.67
  4991.2  575.45  4998.6  574.45    5027  575.45  5027.1  586.45  5061.6  588.67
  5118.7  588.38  5771.6  590.19  5835.5  587.67  6481.1  589.07  6594.4  591.23
  6674.5  589.05  7236.9  599.28  7675.8   602.7  7784.7  606.05  8272.4  620.77
  8397.4  622.63  8586.2  624.15    8918  619.19  9098.9  618.92  9641.1  630.36
#Mann= 9 ,-1 , 0
  1977.3     .05       0    4666      .1       0  4753.4     .12       0
  4991.2     .07       0    5027     .12       0  5061.6      .1       0
  5118.7     .05       0  7675.8     .08       0  7784.7      .1       0
Bank Sta=4991.2,5027
XS Rating Curve= 0 ,0
Exp/Cntr=0.3,0.1

Type RM Length L Ch R = 1 ,400954  ,1582,1582,1582
BEGIN DESCRIPTION:
San Miguel Creek 220.0
END DESCRIPTION:
XS GIS Cut Line= 3
      1990348.56     13571436.46       1986530.8     13571774.54
      1982524.05     13572335.34
#Sta/Elev= 30
  1167.3  632.91    1262  631.45    1361   629.8  1603.4  625.38  1974.9   626.4
  3223.9  608.52  3592.8  603.08  4046.8  607.26    4392  601.94  4776.7  588.89
    4933  582.49  4978.2  586.66  4988.3  584.03  4990.5   573.3  4997.9   572.3
  5026.3   573.3  5033.6  581.72  5053.8   586.2  5089.2   581.2  5110.4   584.9
  6122.5  587.92    6322  583.75  6721.1  588.27  6820.8  591.93  6914.7  598.87
  7320.7  606.24  7840.7  598.96  8532.4  620.67  8830.3  615.58  9045.8  619.68
#Mann= 15 ,-1 , 0
  1167.3      .1       0    1262     .05       0    1361      .1       0
  1974.9     .05       0  3223.9      .1       0  4046.8     .05       0
    4392      .1       0  4776.7     .12       0  4990.5     .07       0
  5026.3     .12       0  5110.4      .1       0  6122.5     .12       0
    6322      .1       0  6721.1     .08       0  6820.8      .1       0
Bank Sta=4990.5,5026.3
XS Rating Curve= 0 ,0
Exp/Cntr=0.3,0.1

Type RM Length L Ch R = 1 ,399372  ,1520,1520,1520
BEGIN DESCRIPTION:
San Miguel Creek 219.0
END DESCRIPTION:
XS GIS Cut Line= 3
      1990101.37     13570558.56       1985850.8     13570474.54
      1981860.86       13571213.
#Sta/Elev= 30
   748.6  620.74  1632.6  608.47  1977.7  610.85    3163  592.09  3180.5  591.85
    3616  587.93  3714.3  588.03  3910.9  583.99  3993.1  587.25  4018.1   583.2
    4086   584.5  4384.5  587.75  4542.4  587.76  4968.3  583.42  4993.3  580.72
  4995.6  571.46  5003.1  570.46  5031.4  571.46  5033.9  578.82  5037.2  580.12
  5086.1  585.69  5593.2  585.87  5669.5  577.93  5799.2  586.76  6099.1   594.8
  6199.7  594.35  6823.8   592.5  7561.1   606.5  8492.9  610.88  9057.7  624.22
#Mann= 14 ,-1 , 0
   748.6     .05       0    3163      .1       0  3180.5     .05       0
    3616      .1       0  3714.3     .16       0  3910.9      .1       0
    4086     .05       0  4384.5      .1       0  4542.4     .12       0
  4995.6     .07       0  5031.4     .12       0  5037.2      .1       0
  6099.1     .08       0  6199.7      .1       0
Bank Sta=4995.6,5031.4
XS Rating Curve= 0 ,0
Exp/Cntr=0.3,0.1

Type RM Length L Ch R = 1 ,397852  ,1115,1115,1115
BEGIN DESCRIPTION:
San Miguel Creek 217.0
END DESCRIPTION:
XS GIS Cut Line= 3
      1989205.97     13568868.76       1986270.8     13569144.54
      1982144.41     13570085.87
#Sta/Elev= 30
  2051.9  623.31  2385.1  621.66  3225.5  608.55  3986.2  607.65  4085.3   606.2
  4385.6  603.56  4737.5   592.6    4878  587.09  4983.2  579.68  4986.1  568.68
  4993.5  567.68    5022  568.68  5022.9   577.2  5039.3  577.06  5054.7  571.28
  5085.4   580.9  5150.3  584.16  5183.7  582.64  5336.7  586.33  5607.5  581.36
  5696.8  582.39  6103.5  585.87  6341.9  580.07    6704  587.48  6805.6   588.3
    8460  600.33  8794.2  607.16  9044.3  612.47    9119  613.68  9232.4  616.24
#Mann= 14 ,-1 , 0
  2051.9      .1       0  3986.2     .08       0  4085.3      .1       0
  4737.5     .16       0    4878     .12       0  4986.1     .07       0
    5022     .12       0  5150.3     .16       0  5696.8      .1       0
    6704     .08       0  6805.6     .05       0  8794.2      .1       0
  9044.3     .05       0    9119      .1       0
Bank Sta=4986.1,5022
XS Rating Curve= 0 ,0
Exp/Cntr=0.3,0.1

Type RM Length L Ch R = 1 ,396737  ,1167,1167,1167
BEGIN DESCRIPTION:
San Miguel Creek 216.0
END DESCRIPTION:
XS GIS Cut Line= 3
       1989137.3     13568152.81      1985783.51     13568211.15
      1981949.89     13568248.29
#Sta/Elev= 30
  1645.7  650.96  2845.7  602.65  3120.7  597.33  3595.1  601.08  3652.7  601.05
  4657.1  594.58  4797.5  588.36  4866.4  584.62  4973.5  577.31    4981  576.99
  4981.3  566.43  4988.8  565.43  5017.2  566.43    5026  576.58    5041  579.19
  5183.5  582.66    5466   581.8  5739.6  582.99    5836  584.06    5871  575.23
  5936.4  579.23  5981.1  585.09  6133.2  583.93  6231.6  583.63    6330  584.16
  6711.1  586.45  7596.1   612.8  8171.2  606.46  8691.2  622.81  8833.8  635.29
#Mann= 16 ,-1 , 0
  1645.7      .1       0  3595.1     .08       0  3652.7      .1       0
  4657.1     .12       0  4797.5     .16       0  4866.4     .12       0
  4973.5      .1       0  4981.3     .07       0  5017.2      .1       0
  5183.5     .05       0    5466      .1       0  5739.6     .12       0
  5936.4     .05       0  6133.2      .1       0  6231.6     .08       0
    6330      .1       0
Bank Sta=4981.3,5017.2
XS Rating Curve= 0 ,0
Exp/Cntr=0.3,0.1

Type RM Length L Ch R = 1 ,395570  ,928,928,928
BEGIN DESCRIPTION:
San Miguel Creek 215.0
END DESCRIPTION:
XS GIS Cut Line= 3
      1989059.19     13567987.89      1986036.54      13567308.8
      1983147.74     13567310.79
#Sta/Elev= 30
    1902  650.08  1961.7  650.34  2170.2  630.58  2555.5  613.65  3446.3  592.05
  3865.8  590.09  4003.1  589.45  4327.7  583.99  4348.2  579.68  4404.6  578.75
  4435.3  583.17  4624.4  584.93  4893.1  581.29  4968.3  576.31  4986.1  565.99
  4993.5  564.99    5022  565.99    5044  577.99  5275.5  581.25  5680.5   579.3
    5814  577.19  5881.8  580.48    6039  583.32  6554.2  581.47  6585.5  581.73
  6652.6   583.3    6829  583.84    7444  605.69    7824  627.09  7888.8  635.39
#Mann= 13 ,-1 , 0
    1902      .1       0  3865.8     .05       0  4003.1      .1       0
  4624.4     .16       0  4893.1     .12       0  4986.1     .07       0
    5022     .12       0  5275.5     .05       0  5680.5      .1       0
  5881.8     .05       0  6554.2     .08       0  6585.5     .05       0
  6652.6      .1       0
Bank Sta=4986.1,5022
XS Rating Curve= 0 ,0
Exp/Cntr=0.3,0.1

Type RM Length L Ch R = 1 ,394642  ,142,142,142
BEGIN DESCRIPTION:
San Miguel Creek 214.0
END DESCRIPTION:
XS GIS Cut Line= 6
      1988624.97     13566774.99      1987908.75     13566596.99
      1987240.35     13566614.35      1986690.91     13566679.33
      1984403.77     13567079.89      1983152.92     13567196.21
#Sta/Elev= 30
  3040.1  620.44  3849.4  590.26  4330.3  584.45    4360  584.07    4528  583.99
  4627.4  581.27  4948.1  579.94  4973.2  574.33  4975.4  566.43  4982.9  565.43
  5011.3  566.43  5013.6  571.83  5018.7  572.96  5057.7  573.54    5218  580.45
    5326  580.43  5562.1  578.56    5727  577.82  5827.3  577.56  5927.5  577.29
  6066.4  576.49  6334.1   578.7  6570.8  578.51  7031.9  579.68  7035.4  579.69
  7299.4  583.21  7575.4  595.37  8292.7  613.55  8508.6  625.99  8578.5  633.57
#Mann= 20 ,-1 , 0
  3040.1      .1       0  4330.3     .08       0    4360     .16       0
    4528      .1       0  4627.4     .08       0  4975.4     .07       0
  5011.3     .08       0  5057.7     .16       0    5218     .12       0
    5326     .08       0  5562.1     .16       0    5727      .1       0
  5827.3     .08       0  5927.5     .05       0  6066.4      .1       0
  6334.1     .08       0  6570.8     .05       0  7031.9     .08       0
  7035.4     .05       0  7575.4      .1       0
Bank Sta=4975.4,5011.3
XS Rating Curve= 0 ,0
Exp/Cntr=0.3,0.1

Type RM Length L Ch R = 1 ,394500  ,375,375,375
BEGIN DESCRIPTION:
Mapping XS 1f2e739d
END DESCRIPTION:
XS GIS Cut Line= 6
      1988646.59     13566714.18      1987900.07      13566458.1
      1987305.45      13566458.1      1986684.79     13566540.57
      1984393.12     13566909.49      1983160.53     13567035.36
#Sta/Elev= 30
  2986.6  620.69  3526.4  600.26  3920.8  587.32  4216.2  582.03  4314.8  581.41
    4707  582.88    4877  580.07  4959.1  576.57  4974.2  573.72  4979.1  566.13
  4986.5  565.13    5015  566.13  5019.7  573.65  5116.5  578.88  5266.9   577.5
  5412.3  575.29  5704.8  579.43  5785.5  579.18    5913  575.28  7102.5  583.96
  7197.8  588.85    7288  605.62  7350.9  601.75  7434.5  603.07  7513.3  610.28
  7810.8  607.74  8092.1  616.67  8248.7  630.32  8399.5  623.83  8557.3  628.78
#Mann= 19 ,-1 , 0
  2986.6      .1       0  3526.4     .08       0  3920.8     .05       0
  4216.2     .08       0  4314.8     .05       0    4707     .08       0
    4877     .12       0  4979.1     .07       0    5015     .12       0
  5116.5     .16       0  5266.9     .08       0  5412.3      .1       0
  5704.8     .16       0  5785.5     .08       0    5913      .1       0
  7350.9     .08       0  7513.3      .1       0  7810.8     .08       0
  8092.1      .1       0
Bank Sta=4979.1,5015
XS Rating Curve= 0 ,0
Exp/Cntr=0.3,0.1

Type RM Length L Ch R = 1 ,394125  ,837,837,837
BEGIN DESCRIPTION:
San Miguel Creek 213.0
END DESCRIPTION:
XS GIS Cut Line= 4
      1988663.95     13566653.41      1987904.41     13566358.28
        1986625.       13566175.      1984067.65     13566605.66
#Sta/Elev= 30
  2888.4  620.41  3182.1  611.76    3337     606  3478.2   602.3    3703  591.13
  3833.2  589.55  4641.7  580.65  4740.7  580.76  4937.7  576.62    4963  572.26
  4965.2  564.77  4972.6  563.77  5001.1  564.77  5003.3  570.08  5033.8  576.46
  5074.3  578.46  5280.6  577.29  5386.7  569.55  5416.9   576.8  5447.2  578.11
    5717  575.83  5991.5   585.6  6292.1  597.47  6498.9  613.75  6589.7  608.75
  6680.5  597.53  6743.5  598.31  7225.3  616.62  7346.3  627.14  7589.1  633.81
#Mann= 11 ,-1 , 0
  2888.4      .1       0  3182.1     .05       0    3337     .08       0
  3478.2      .1       0  3833.2     .05       0  4641.7     .08       0
  4740.7     .12       0  4965.2     .07       0  5001.1     .12       0
  5280.6     .16       0  5991.5      .1       0
Bank Sta=4965.2,5001.1
XS Rating Curve= 0 ,0
Exp/Cntr=0.3,0.1

Type RM Length L Ch R = 1 ,393288  ,1113,1113,1113
BEGIN DESCRIPTION:
San Miguel Creek 212.0
END DESCRIPTION:
XS GIS Cut Line= 3
      1988594.52     13566384.32      1986599.83     13565469.42
      1984784.42     13565642.07
#Sta/Elev= 30
  2805.5  614.47  3165.8  603.28  3341.1  604.09  3396.3  601.71  3482.9  593.79
  3570.5   588.8  3705.2  584.39  3973.9  579.32  4188.4  578.72  4780.3  582.06
  4964.7  578.39  4980.6   570.5  4981.2  562.37  4988.7  561.37  5017.2  562.37
  5017.4  567.13  5042.5  574.78  5087.1  577.17  5131.1  577.97  5324.7  575.57
  5358.9  572.64  5373.7  575.49  5400.9  575.54  5474.5  578.04  5499.6  581.01
  5663.8  586.51  5809.8  593.12  6207.8  612.18  6468.9     619  6823.6  631.97
#Mann= 10 ,-1 , 0
  2805.5      .1       0  3482.9     .05       0  4780.3     .12       0
  4981.2     .07       0  5017.2     .12       0  5087.1     .16       0
  5131.1     .12       0  5400.9      .1       0  5663.8     .05       0
  5809.8      .1       0
Bank Sta=4981.2,5017.2
XS Rating Curve= 0 ,0
Exp/Cntr=0.3,0.1

Type RM Length L Ch R = 1 ,392175  ,1017,1017,1017
BEGIN DESCRIPTION:
San Miguel Creek 211.0
END DESCRIPTION:
XS GIS Cut Line= 4
      1988455.61     13564570.08      1986580.62     13564778.42
      1986199.83     13564915.95      1984779.69      13565533.5
#Sta/Elev= 30
  2708.6  599.81  2844.4  599.21  3211.9   589.2    3394  587.08  3587.1  580.06
  3798.4   576.9    4250  576.62  4349.3  576.68  4448.6  577.08  4660.1  577.22
  4676.6   577.5  4949.3  574.67  4983.2  570.49  4989.7  559.86  4997.2  558.86
  5025.7  559.86  5029.8   572.9  5075.8  575.95  5097.9  575.74  5121.4  579.45
  5215.6  581.03  5391.6  587.31  5540.8   594.8  5541.2  594.82  5591.4  600.06
  5607.7  598.75  5660.8  602.88  5864.7  605.87  6267.5   624.2  6548.6  629.02
#Mann= 15 ,-1 , 0
  2708.6     .05       0  3211.9      .1       0    3394     .05       0
    4250      .1       0  4349.3     .05       0  4448.6     .12       0
  4660.1      .1       0  4676.6     .12       0  4989.7     .07       0
  5025.7     .12       0  5075.8      .1       0  5215.6     .05       0
  5391.6      .1       0  5540.8     .05       0  5541.2      .1       0
Bank Sta=4989.7,5025.7
XS Rating Curve= 0 ,0
Exp/Cntr=0.3,0.1

Type RM Length L Ch R = 1 ,391158  ,1194,1194,1194
BEGIN DESCRIPTION:
San Miguel Creek 210.0
END DESCRIPTION:
XS GIS Cut Line= 4
       1988685.3      13564182.1       1986120.8     13563924.54
      1985669.53      13564145.1      1984324.49     13565498.81
#Sta/Elev= 30
  2422.6  599.62  2641.3   599.6  3192.9  587.34  3995.2  577.84    4093  573.35
  4268.5  574.88    4367  574.89  4460.9  575.26  4630.7  575.56  4790.3   576.6
  4892.8  573.98    4933  568.03  4968.1  573.12  4983.2  570.71  4985.8  560.65
  4993.3  559.65  5021.8  560.65  5023.5  566.64  5031.5  571.91  5064.1   570.9
  5158.6  575.98  5286.5  576.32  5479.4  577.16  5887.3     598  6265.6  604.05
  6594.4  602.39  6940.9  617.42  7213.1  610.33  7301.5  613.12  7410.6  622.85
#Mann= 10 ,-1 , 0
  2422.6     .05       0  4268.5      .1       0    4367     .05       0
  4460.9      .1       0  4630.7     .16       0  4790.3     .12       0
  4985.8     .07       0  5021.8     .12       0  5064.1     .16       0
  5286.5      .1       0
Bank Sta=4985.8,5021.8
XS Rating Curve= 0 ,0
Exp/Cntr=0.3,0.1

Type RM Length L Ch R = 1 ,389964  ,676,676,676
BEGIN DESCRIPTION:
San Miguel Creek 209.0
END DESCRIPTION:
XS GIS Cut Line= 3
      1988904.11     13563124.81       1985530.8     13563024.54
      1983831.16     13563682.09
#Sta/Elev= 30
  1625.2  596.37  2124.1  589.72  2547.2  593.04  3452.1  579.44  3687.7  579.51
  3772.8  574.55  3848.9  577.51  3947.2  574.27  4092.9  572.42  4107.9  569.25
  4122.9  572.44  4157.9  570.42    4338   573.6  4660.3  573.47  4758.2  570.79
  4973.3  570.84  4993.3  568.23  4997.9  565.19    4998  558.82  5005.5  557.82
  5034.1  558.82  5035.7  566.61  5046.4  573.39  5137.8  573.54  5244.8  573.04
  5400.3  578.16  5900.3  605.56  6125.2  614.76  6400.5  612.41  6822.4  619.45
#Mann= 9 ,-1 , 0
  1625.2     .05       0  3452.1      .1       0  3848.9     .05       0
  3947.2     .16       0  4660.3     .12       0    4998     .07       0
  5034.1     .12       0  5137.8      .1       0  5900.3     .05       0
Bank Sta=4998,5034.1
XS Rating Curve= 0 ,0
Exp/Cntr=0.3,0.1

Type RM Length L Ch R = 1 ,389288  ,999,999,999
BEGIN DESCRIPTION:
San Miguel Creek 208.0
END DESCRIPTION:
XS GIS Cut Line= 4
      1988013.39     13562390.43        1985675.       13562425.
      1984816.82     13562551.46      1983789.72     13563431.89
#Sta/Elev= 30
    2647  595.46  3958.8   585.8  4057.2  585.17  4155.6   582.9  4259.8  580.01
  4478.1  570.55  4513.1  565.71  4543.1  569.38  4570.1  569.31  4888.1   572.6
  4938.1  568.78  4958.1  568.88  4968.1  564.31  4970.1  559.38  4977.7  558.38
  5006.2  559.38    5018  568.77  5020.5  566.92  5023.6  570.53  5033.7  572.42
    5166  573.34    5535  572.66  5695.7  570.57  5837.2  573.25    6059  588.23
  6292.2  592.85  6690.1   595.6  6821.2  602.36  6878.3  606.99  7205.9  616.87
#Mann= 11 ,-1 , 0
    2647     .05       0  3958.8      .1       0  4057.2     .08       0
  4155.6      .1       0  4259.8     .16       0  4570.1     .12       0
  4970.1     .07       0  5006.2     .12       0    5166     .16       0
    5535      .1       0  6292.2     .05       0
Bank Sta=4970.1,5006.2
XS Rating Curve= 0 ,0
Exp/Cntr=0.3,0.1

Type RM Length L Ch R = 1 ,388289  ,752,752,752
BEGIN DESCRIPTION:
San Miguel Creek 207.0
END DESCRIPTION:
XS GIS Cut Line= 4
      1987924.98       13561575.        1985925.       13561575.
      1984816.82     13561843.12      1982699.36     13562703.99
#Sta/Elev= 30
  3016.5   600.3    3499  593.19    3854  584.63  4138.9  580.25  4410.2  577.46
    4464  576.68  4508.6  573.17  4703.6  571.87    4754  570.42    4769  572.11
    4829  568.86  4913.9  570.13    4964   569.5    4969  568.69    4979  561.24
  4987.5  559.56  4990.9   559.5  4998.4   558.4    5027   559.5  5037.4   568.2
  5049.9  571.32  5101.7  571.08  5203.7  570.74  5481.8  573.81  6281.9  569.77
  6359.5  572.63    7184  584.24    7726  594.67  8142.3  599.33  8442.4  608.74
#Mann= 11 ,-1 , 0
  3016.5     .05       0  4138.9      .1       0  4410.2     .05       0
  4508.6      .1       0  4703.6     .12       0  4913.9     .16       0
  4987.5     .12       0  4990.9     .07       0    5027     .12       0
  5101.7     .16       0  5203.7     .05       0
Bank Sta=4990.9,5027
XS Rating Curve= 0 ,0
Exp/Cntr=0.3,0.1

Type RM Length L Ch R = 1 ,387537  ,787,787,787
BEGIN DESCRIPTION:
San Miguel Creek 206.0
END DESCRIPTION:
XS GIS Cut Line= 4
      1987511.27     13560905.62       1986180.8     13560913.65
      1985080.71     13561030.62      1982615.43     13562242.65
#Sta/Elev= 30
  3669.5   595.1  4538.3  586.13  4628.7  583.39  4727.1  581.01  4825.4  577.25
  4968.3  570.39  4973.3  569.55  4975.2  554.96  4982.7  553.86  5011.3  554.96
  5011.8  557.18  5028.5  568.46  5068.7  564.61  5088.8  567.99  5121.6  569.35
  5220.9  569.01  5330.1  566.84    5721  572.77  6260.3   573.7    6755  569.68
  6928.9  569.58  7118.5     577  7364.5   583.1  7881.5  584.27  8392.8  589.51
  8687.7  593.69  8766.4  596.32  8795.4  599.59  8822.6  595.72  8853.4  596.32
#Mann= 10 ,-1 , 0
  3669.5     .05       0  4628.7      .1       0  4727.1     .05       0
  4825.4     .12       0  4975.2     .07       0  5011.3     .12       0
  5121.6      .1       0  5220.9     .05       0    6755      .1       0
  7118.5     .05       0
Bank Sta=4975.2,5011.3
XS Rating Curve= 0 ,0
Exp/Cntr=0.3,0.1

Type RM Length L Ch R = 1 ,386750  ,1349,1349,1349
BEGIN DESCRIPTION:
Mapping XS 8bca09ed
END DESCRIPTION:
XS GIS Cut Line= 4
      1987820.32     13560108.75      1986101.55     13560160.83
       1985094.6     13560317.08      1982364.38      13561747.5
#Sta/Elev= 30
  3299.7  595.16  4165.9  584.08  4333.5   585.4  4642.9     579  4741.4  575.82
  4839.9  572.89  4973.3  566.06  4988.3  559.87  4990.3  551.57  4997.8  550.47
  5026.4  551.57  5028.4  563.21  5033.5  566.61  5087.5  566.78  5241.2  566.39
  5502.2  570.19  6015.1  572.33  6303.1  572.31    6637  568.02  6887.5  568.82
  6928.8  574.21  6939.9  573.56  6959.1  566.23  6970.1   564.6  7036.3  564.36
  7073.6  573.39  7167.1  573.62    7651  577.94  8469.7  591.21  9120.5  594.04
#Mann= 10 ,-1 , 0
  3299.7     .05       0  4642.9      .1       0  4741.4     .16       0
  4839.9     .12       0  4990.3     .07       0  5026.4     .12       0
  5087.5     .16       0  5241.2     .05       0    6637      .1       0
  7167.1     .05       0
Bank Sta=4990.3,5026.4
XS Rating Curve= 0 ,0
Exp/Cntr=0.3,0.1

Type RM Length L Ch R = 1 ,385401  ,1206,1206,1206
BEGIN DESCRIPTION:
San Miguel Creek 205.0
END DESCRIPTION:
XS GIS Cut Line= 3
      1987769.53     13559797.99       1986110.8     13559024.54
      1981547.76     13559838.12
#Sta/Elev= 30
  3169.8  591.61  3999.6  572.61  4437.5  568.55  4562.6  566.67    4586  566.38
  4601.6  563.43  4611.9  563.28  4628.5  566.09  4669.6  566.62  4755.4  567.17
  4834.3   564.2  4909.9  567.15  4928.5  566.44    4977  563.26  4981.6  561.61
  4983.7  548.52  4991.2  547.42  5019.8  548.52  5023.7  559.35  5033.8   562.7
    5192  568.44  5372.3  569.95  5745.3  566.02  5831.2  568.07  6262.9  570.64
  6902.5  566.61  8462.3  576.29  9048.1  582.85  9359.7  588.91    9635   592.1
#Mann= 10 ,-1 , 0
  3169.8     .05       0  4437.5      .1       0  4562.6     .12       0
  4601.6     .16       0  4669.6     .12       0  4983.7     .07       0
  5019.8     .12       0    5192      .1       0  6902.5     .05       0
  8462.3      .1       0
Bank Sta=4983.7,5019.8
XS Rating Curve= 0 ,0
Exp/Cntr=0.3,0.1

Type RM Length L Ch R = 1 ,384195  ,1755,1755,1755
BEGIN DESCRIPTION:
San Miguel Creek 204.0
END DESCRIPTION:
XS GIS Cut Line= 3
      1988474.98     13558474.99       1986360.8     13557954.54
      1981691.78      13559153.9
#Sta/Elev= 30
  2822.7  593.62  4200.1  581.51  4686.2  570.28  4933.9  564.37  4978.7  561.05
  4982.8  558.58  4985.9  546.67  4993.4  545.57    5022  546.67  5024.3  561.21
  5042.1  563.89  5346.3  564.67  5553.1  565.07  5571.4  565.09  5860.4  564.96
  5887.4  558.64  5907.8  558.32  6032.7   564.3  6228.6  562.86  6474.7  568.38
    7026  567.63  7084.8  566.61  7190.5  565.45  7231.8  562.91  7426.1  572.16
  7604.4  568.09  8605.9  573.26  8881.7  576.96  9380.7  592.46  9820.6  597.07
#Mann= 15 ,-1 , 0
  2822.7     .05       0  4686.2      .1       0  4933.9     .12       0
  4985.9     .07       0    5022     .12       0  5346.3     .16       0
  5553.1     .12       0  5571.4     .16       0  6032.7      .1       0
    7026     .16       0  7084.8      .1       0  7190.5     .16       0
  7426.1      .1       0  7604.4     .05       0  8605.9      .1       0
Bank Sta=4985.9,5022
XS Rating Curve= 0 ,0
Exp/Cntr=0.3,0.1

Type RM Length L Ch R = 1 ,382440  ,1517,1517,1517
BEGIN DESCRIPTION:
San Miguel Creek 203.0
END DESCRIPTION:
XS GIS Cut Line= 3
      1988472.62     13558226.79       1985510.8     13556824.54
      1982459.64      13556522.2
#Sta/Elev= 30
    1723  591.62  3524.5  565.53  3783.8  561.43  4162.8  568.29  4582.7  563.87
  4757.2  562.78  4959.4  560.61  4977.2  555.72    4979  545.07  4986.6  543.97
  5015.2  545.07  5018.4  555.69  5023.4  559.44  5033.5  560.23    5144  559.59
  5164.1  562.16  5334.9  565.14  5445.5  563.16  6204.6  567.13  7093.5  567.03
  7340.5  573.84  7520.6  579.61  7632.9  589.06  7691.4  590.56  7721.6  588.52
    7807  598.36  7885.2  594.78  7927.6   596.1  7992.9   604.9  8066.1  609.12
#Mann= 8 ,-1 , 0
    1723     .05       0  3524.5      .1       0  4582.7     .16       0
  4757.2     .12       0    4979     .07       0  5015.2     .12       0
  6204.6     .05       0  7340.5      .1       0
Bank Sta=4979,5015.2
XS Rating Curve= 0 ,0
Exp/Cntr=0.3,0.1

Type RM Length L Ch R = 1 ,380923  ,1311,1311,1311
BEGIN DESCRIPTION:
San Miguel Creek 201.0
END DESCRIPTION:
XS GIS Cut Line= 4
      1988978.31     13556435.36       1986490.8     13555754.54
      1985714.39       13555575.      1982694.27     13555697.48
#Sta/Elev= 30
    2421  583.43  2616.8  582.88    3906   578.5    4658  556.59  4939.3   560.2
  4972.3  555.99  4977.1  553.29  4978.8  542.12  4986.4  541.02    5015  542.12
  5018.2  551.67  5023.9  555.77  5042.1  558.84  5193.1  558.95    5242  556.55
    5266  551.12  5314.4   557.6  5505.4  561.35  5522.4  561.37  6504.4  563.77
  6974.8  559.67    7320  564.75  7935.5  578.33  8105.7  597.46  8215.8  581.45
    8491  588.12  8556.1  594.54  8571.1  592.26  8691.2  606.46  8819.5  613.56
#Mann= 10 ,-1 , 0
    2421      .1       0  2616.8     .05       0    3906      .1       0
  4939.3     .12       0  4978.8     .07       0    5015     .12       0
  5193.1     .16       0  5314.4      .1       0  5505.4     .16       0
  5522.4      .1       0
Bank Sta=4978.8,5015
XS Rating Curve= 0 ,0
Exp/Cntr=0.3,0.1

Type RM Length L Ch R = 1 ,379612  ,931,931,931
BEGIN DESCRIPTION:
San Miguel Creek 200.0
END DESCRIPTION:
XS GIS Cut Line= 3
       1989030.4     13555306.89        1986525.       13554925.
      1982745.68     13555558.61
#Sta/Elev= 30
  2461.4  587.12  3187.6   578.5  3503.1  579.55  4317.3   558.1  4441.9  553.58
    4496   556.5  4905.4   559.5    4964  557.63  4988.2  551.14  4990.3   540.4
  4997.9   539.3  5026.5   540.4  5028.7   551.6  5064.2  558.63  5128.5  558.71
  5454.6  562.46  6169.4  558.59  6682.1  559.85  6787.9  559.66  7223.9  565.87
  7323.5  573.67  7626.8  589.06  7796.8  585.72  7927.5  592.04  8018.5   590.6
  8112.1  595.14  8200.5  588.21  8261.2  587.52  8628.2   597.8  8827.8  607.47
#Mann= 9 ,-1 , 0
  2461.4      .1       0  4317.3     .12       0    4496      .1       0
  4905.4     .12       0  4990.3     .07       0  5026.5     .12       0
  5128.5      .1       0  6682.1     .12       0  6787.9      .1       0
Bank Sta=4990.3,5026.5
XS Rating Curve= 0 ,0
Exp/Cntr=0.3,0.1

Type RM Length L Ch R = 1 ,378681  ,928,928,928
BEGIN DESCRIPTION:
San Miguel Creek 199.0
END DESCRIPTION:
XS GIS Cut Line= 3
      1989030.32     13554612.43        1986425.       13554075.
      1982815.11     13555358.96
#Sta/Elev= 30
  2299.2  583.82  3180.2  569.86  3921.5  570.13  4113.7  562.44  4293.4  553.84
  4484.6  555.35  4612.6  558.72  4812.2  555.88  4886.5  557.04    4962  553.54
  4967.3  551.22  4969.5  537.44    4977  536.34  5005.7  537.44  5009.8  548.73
  5025.7  555.81  5120.4  556.85  5204.6  558.09  5225.9   558.4  5752.3  558.46
  6825.7  559.39  7189.1  561.59  7337.3  563.56  7366.1  564.16  7809.2  572.23
  7868.2  574.46  7886.3  578.68  7927.2  573.41  8599.9  595.11  8790.8   610.4
#Mann= 15 ,-1 , 0
  2299.2      .1       0  4113.7     .12       0  4484.6      .1       0
  4612.6     .16       0  4812.2     .12       0  4969.5     .07       0
  5005.7     .12       0  5120.4     .16       0  5204.6      .1       0
  5225.9     .16       0  5752.3      .1       0  6825.7     .07       0
  7189.1     .12       0  7337.3     .07       0  7366.1      .1       0
Bank Sta=4969.5,5005.7
XS Rating Curve= 0 ,0
Exp/Cntr=0.3,0.1

Type RM Length L Ch R = 1 ,377753  ,1141,1141,1141
BEGIN DESCRIPTION:
San Miguel Creek 198.0
END DESCRIPTION:
XS GIS Cut Line= 3
      1988874.97       13553575.        1986475.       13553275.
      1983024.25     13554273.65
#Sta/Elev= 30
  2589.4  584.87  2692.6  584.73  2912.8  582.82  3599.7  574.66  3629.9  571.45
    3640  573.42  3803.1  571.39  3942.4  569.69  4196.3  564.32  4425.8  555.93
  4486.5  553.03    4552  556.19  4647.8  552.55  4733.4  556.15  4899.7  555.59
  4965.6  551.34  4980.3     548  4982.4  539.35  4989.9  538.25  5018.6  539.35
  5021.1  551.05  5036.7  554.85  5225.2  553.93  5743.7  558.26  6685.3  559.63
    6693  559.59  7602.8  563.57  7941.8     575  8123.3  585.79  8600.4  592.62
#Mann= 13 ,-1 , 0
  2589.4     .05       0  2692.6      .1       0  2912.8     .05       0
  3803.1      .1       0  3942.4     .05       0  4196.3     .16       0
  4425.8     .12       0  4965.6     .16       0  4982.4     .07       0
  5018.6     .12       0  5225.2      .1       0  6685.3     .05       0
    6693      .1       0
Bank Sta=4982.4,5018.6
XS Rating Curve= 0 ,0
Exp/Cntr=0.3,0.1

Type RM Length L Ch R = 1 ,376612  ,966,966,966
BEGIN DESCRIPTION:
San Miguel Creek 197.0
END DESCRIPTION:
XS GIS Cut Line= 3
       1988995.6     13552676.67      1985928.84     13552390.32
      1983032.13     13553466.59
#Sta/Elev= 30
  1919.9  578.31  2184.1   572.4  2289.6  575.35  2888.2   576.1    2990  575.19
    3073  573.76  3098.1  575.64  3143.3  572.92  3600.3  567.71    4007  552.43
  4127.6  557.24  4619.6  554.09  4780.6  553.02  4951.6  551.23  4976.2  548.54
  4988.7  538.91  4996.2  537.81  5024.9  538.91  5026.6  552.28  5044.5  554.03
  5454.8  551.17  5616.9  552.64  5745.6  556.99  5984.7  557.36  6148.8  560.15
  6779.8  577.53  6932.3  585.18  7110.2  579.77  7397.8  585.06  8090.2  587.76
#Mann= 9 ,-1 , 0
  1919.9      .1       0  2888.2     .05       0    2990      .1       0
  4619.6     .16       0  4780.6     .12       0  4988.7     .07       0
  5024.9     .12       0  5984.7     .05       0  6148.8      .1       0
Bank Sta=4988.7,5024.9
XS Rating Curve= 0 ,0
Exp/Cntr=0.3,0.1

Type RM Length L Ch R = 1 ,375646  ,567,567,567
BEGIN DESCRIPTION:
San Miguel Creek 196.0
END DESCRIPTION:
XS GIS Cut Line= 3
      1988934.83     13551652.37      1985479.63     13551588.24
      1983040.82     13552858.95
#Sta/Elev= 30
  1544.2  580.16    2087  572.64  2521.7  566.61  2701.7  569.83  2770.1  568.45
  2888.8  566.72  2951.8  566.04  2971.8  562.44  3289.9  556.23  3487.1     552
  4208.6  555.19    4635  557.08  4779.5  553.34  4862.1  549.13  4962.1  550.37
  4977.1   544.4  4986.4   537.1    4994     536  5022.6   537.1  5023.8  547.24
    5068  552.39  5120.4  553.67  5223.2  552.02  5354.9  552.74  5609.1   550.4
  5968.1  561.96    6084  569.14  6376.6  573.88  6616.9  580.21    7750  578.74
#Mann= 12 ,-1 , 0
  1544.2     .05       0    2087      .1       0  2770.1     .05       0
  2888.8      .1       0  3289.9     .16       0  3487.1      .1       0
  4208.6     .16       0  4779.5     .12       0  4986.4     .07       0
  5022.6     .12       0  5223.2     .16       0  5354.9      .1       0
Bank Sta=4986.4,5022.6
XS Rating Curve= 0 ,0
Exp/Cntr=0.3,0.1

Type RM Length L Ch R = 1 ,375079  ,236,236,236
BEGIN DESCRIPTION:
Mapping XS d471e6fc
END DESCRIPTION:
XS GIS Cut Line= 3
      1988943.53     13550775.63      1985427.94     13551027.37
       1982224.9     13551374.58
#Sta/Elev= 30
  1484.2  578.06  1567.3  576.64  1893.2  569.17  1999.7  566.99  2068.6  565.35
  2677.9  562.01  2776.7  562.27  3254.8   555.6  3555.5  550.92  3693.4  552.37
  4160.3  554.58  4417.9  558.02  4844.3   551.2  4976.2   547.7  4979.2  545.89
  4981.1  537.69  4988.7  536.59  5017.3  537.69  5019.3  546.41  5024.3  548.22
  5064.6  551.24  5228.9  549.27  5602.9  549.05  5758.6  551.08  5949.7  558.75
  6131.8  558.87  6467.7  560.68  6593.5  564.73  7704.9  567.37  8230.6     579
#Mann= 16 ,-1 , 0
  1484.2      .1       0  1567.3     .05       0  1893.2      .1       0
  1999.7     .05       0  2068.6      .1       0  2677.9     .08       0
  2776.7      .1       0  3254.8     .16       0  3693.4      .1       0
  4160.3     .16       0  4844.3     .12       0  4981.1     .07       0
  5017.3     .12       0  5228.9      .1       0  5602.9     .16       0
  6131.8      .1       0
Bank Sta=4981.1,5017.3
XS Rating Curve= 0 ,0
Exp/Cntr=0.3,0.1

Type RM Length L Ch R = 1 ,374843  ,1073,1073,1073
BEGIN DESCRIPTION:
Mapping XS 5c4f15a8
END DESCRIPTION:
XS GIS Cut Line= 3
      1988969.58     13550558.62      1985436.62     13550792.99
      1982207.45     13551131.53
#Sta/Elev= 30
  1472.3  577.54  1871.7  570.43  1894.5  570.46  2092.1  565.72  2346.3  560.33
  2881.1  558.57    2981  558.29  3778.8  552.18  3890.5   551.2  3959.8  549.85
  4462.6  554.28  4899.8  549.71  4956.5  548.13  4977.1  547.62    4979  538.73
  4986.6  537.63  5015.2  538.73    5031  547.15  5074.3  550.77  5228.3  549.05
  5253.5  545.01  5268.5  549.06  5389.2  547.39  5467.2  549.84  5658.2  551.56
    5750  552.79  6326.9  560.84  7535.9  567.54  7673.5  568.47  8259.9  577.67
#Mann= 19 ,-1 , 0
  1472.3      .1       0  1871.7     .08       0  1894.5     .05       0
  2092.1      .1       0  2881.1     .05       0    2981      .1       0
  3778.8     .12       0  3890.5      .1       0  4462.6     .16       0
  4899.8     .05       0  4956.5     .12       0    4979     .07       0
  5015.2     .12       0  5074.3     .16       0  5467.2      .1       0
  5658.2     .05       0    5750      .1       0  7535.9     .05       0
  7673.5      .1       0
Bank Sta=4979,5015.2
XS Rating Curve= 0 ,0
Exp/Cntr=0.3,0.1

Type RM Length L Ch R = 1 ,373770  ,1258,1258,1258
BEGIN DESCRIPTION:
San Miguel Creek 194.0
END DESCRIPTION:
XS GIS Cut Line= 3
      1988995.64     13550194.03       1985110.8     13550134.54
      1982077.24      13550966.6
#Sta/Elev= 30
  1114.7  570.65  1522.9  566.93  2000.8   558.4  2267.5  557.16  3694.6  551.25
  3908.2  550.44  3938.2  545.12  3963.2  544.27  3998.2  544.87  4028.2  551.42
  4343.2  546.39  4503.2  550.82    4794  550.82  4970.3  549.34  4983.3  547.75
  4985.8  534.15  4993.3  533.05    5022  534.15  5024.2  542.24  5038.3  546.36
  5138.2  545.31  5164.1  549.85  5259.5  553.78  6076.6  562.97  6625.5  560.33
  6986.5  564.04  7077.3  562.02  7253.4  566.32  7356.2  568.07  8145.6  578.99
#Mann= 10 ,-1 , 0
  1114.7      .1       0  2000.8     .12       0  2267.5      .1       0
  3694.6     .16       0    4794     .12       0  4985.8     .07       0
    5022     .12       0  5259.5      .1       0  7253.4     .05       0
  7356.2      .1       0
Bank Sta=4985.8,5022
XS Rating Curve= 0 ,0
Exp/Cntr=0.3,0.1

Type RM Length L Ch R = 1 ,372512  ,1245,1245,1245
BEGIN DESCRIPTION:
San Miguel Creek 193.0
END DESCRIPTION:
XS GIS Cut Line= 3
      1988144.91     13548839.87       1985150.8     13549054.54
      1981974.99     13550625.01
#Sta/Elev= 30
  1998.2  574.49  2306.4  575.09  2632.2  564.23  3208.7  559.66  3484.8  547.54
  3529.5  544.04  3714.3  547.76  3836.5   546.9  4206.1  546.84  4304.9  545.23
  4431.2   546.2  4888.7  548.86  4968.2  544.54  4978.2  539.29  4979.8  532.76
  4987.3  531.66    5016  532.76  5020.4  542.91  5026.2  545.21  5059.8  540.26
  5210.2  548.27  5414.6  550.47  5940.8  559.14  6515.3  559.29  6882.7  551.67
  6978.3   557.1  7559.7  563.97  7671.1  566.58  8360.6  584.92  8542.9  584.51
#Mann= 14 ,-1 , 0
  1998.2      .1       0  3484.8     .12       0  3714.3      .1       0
  3836.5     .05       0  4206.1     .12       0  4304.9      .1       0
  4431.2     .16       0  4888.7     .12       0  4979.8     .07       0
    5016     .12       0  5210.2     .16       0  5414.6      .1       0
  7559.7     .08       0  7671.1      .1       0
Bank Sta=4979.8,5016
XS Rating Curve= 0 ,0
Exp/Cntr=0.3,0.1

Type RM Length L Ch R = 1 ,371267  ,175,175,175
BEGIN DESCRIPTION:
San Miguel Creek 191.0
END DESCRIPTION:
XS GIS Cut Line= 4
      1987680.49     13548283.81       1985180.8     13547904.54
      1984345.86     13547790.92      1981721.36     13549213.12
#Sta/Elev= 30
  2471.7  576.28  2722.5  574.83  3328.6  557.28  3730.9  558.69  4108.2  545.09
    4165   549.2  4331.8  545.78  4416.7  538.87  4509.9  543.49  4589.3  543.23
  4840.2   544.3  4978.1   543.8  4983.1     543  4990.3  531.61  4997.8  530.51
  5026.5  531.61  5028.6  543.05  5032.4  543.93  5127.2  544.81  5385.9  543.98
  5849.4  548.74  5898.9  548.91  6227.1  549.31  6232.5   549.3  6340.9  548.76
  6393.1  548.95  7244.8  549.77  7601.1  555.35  7706.5  557.03  8827.7  578.44
#Mann= 16 ,-1 , 0
  2471.7      .1       0  4509.9     .12       0  4589.3      .1       0
  4840.2     .12       0  4990.3     .07       0  5026.5     .12       0
  5127.2     .16       0  5385.9      .1       0  5849.4     .16       0
  5898.9      .1       0  6227.1     .16       0  6232.5      .1       0
  6340.9     .16       0  6393.1      .1       0  7601.1     .05       0
  7706.5      .1       0
Bank Sta=4990.3,5026.5
XS Rating Curve= 0 ,0
Exp/Cntr=0.3,0.1

Type RM Length L Ch R = 1 ,371092  ,959,959,959
BEGIN DESCRIPTION:
Mapping XS 94d7856f
END DESCRIPTION:
XS GIS Cut Line= 5
      1987704.97     13548121.04      1985861.64     13547834.78
       1985120.8     13547754.54      1984322.83     13547606.18
      1981759.39     13549043.02
#Sta/Elev= 30
  2389.4  575.22  2629.7  577.11  2670.2  571.51  2695.5  575.92    3247  562.54
  3505.8  563.58  3959.1  550.06    4158  555.52    4601   538.4  4766.5  544.36
  4949.9  543.82  4988.2  538.38  4990.3  531.25  4997.9  530.15  5026.5  531.25
  5028.8  538.77  5033.9  540.49  5068.2  544.31    5124   545.1  5252.4  543.79
  5322.9  542.34  5521.8  547.27  5857.5  548.89  6016.6  549.18  6330.9   548.6
  7300.8  549.63  7657.8  555.08  7772.5  557.06  7884.6  558.96  8750.3  584.89
#Mann= 15 ,-1 , 0
  2389.4      .1       0  4766.5     .12       0  4990.3     .07       0
  5026.5     .12       0  5068.2     .16       0    5124      .1       0
  5252.4     .16       0  5322.9      .1       0  5521.8     .05       0
  5857.5      .1       0  6016.6     .16       0  6330.9      .1       0
  7657.8     .08       0  7772.5     .05       0  7884.6      .1       0
Bank Sta=4990.3,5026.5
XS Rating Curve= 0 ,0
Exp/Cntr=0.3,0.1

Type RM Length L Ch R = 1 ,370133  ,1251,1251,1251
BEGIN DESCRIPTION:
San Miguel Creek 190.0
END DESCRIPTION:
XS GIS Cut Line= 3
      1986416.64     13546818.12        1984875.       13547025.
      1981690.09     13548823.33
#Sta/Elev= 30
  3441.8  575.34  3940.4  562.41  4620.1  550.96  4719.6  551.09  4828.3  548.65
  4916.8  543.21  4984.6   539.8  4989.7  538.59  4989.9  530.25  4997.5  529.05
  5026.2  530.25  5026.9  540.62  5029.7  541.87    5229  542.47  5283.2  540.57
  5312.8  537.05  5345.3  541.13  5438.9  545.16  5631.7   548.7  6119.6  547.91
  7067.2  548.39  7471.1  552.27  7586.1  552.72  7874.6   562.5  8022.6  563.99
    8046  562.39  8212.5  567.94    8391  574.78  8402.4   574.8  8654.8  585.02
#Mann= 14 ,-1 , 0
  3441.8      .1       0  4719.6     .16       0  4916.8     .12       0
  4989.9     .07       0  5026.2     .12       0  5438.9     .05       0
  6119.6      .1       0  7471.1     .05       0  7586.1      .1       0
  8022.6     .05       0    8046     .08       0  8212.5     .05       0
    8391     .08       0  8402.4      .1       0
Bank Sta=4989.9,5026.2
XS Rating Curve= 0 ,0
Exp/Cntr=0.3,0.1

Type RM Length L Ch R = 1 ,368882  ,1351,1351,1351
BEGIN DESCRIPTION:
San Miguel Creek 189.0
END DESCRIPTION:
XS GIS Cut Line= 3
      1986976.56     13546101.98       1984250.8     13546074.54
      1980534.51     13548337.57
#Sta/Elev= 30
  2274.1  578.13  2588.2  576.74  3548.2   554.1  4123.3  548.22    4495  547.99
  4713.3   547.7  4859.1  542.72  4978.3   540.3  4979.7  530.18  4987.3  528.98
    5016  530.18  5022.2  534.34  5051.3  535.58  5066.8  540.78  5077.4  541.13
  5288.5  542.57  5575.4  538.79  5589.8  535.89  5608.3  536.25  5729.2  542.72
  5856.1  545.82  6816.8  543.91  7097.2   545.8    7230  546.72    7332  547.68
  7410.2  548.68    7886  558.43  8203.7  560.57  9271.6  569.62  9351.1  570.59
#Mann= 13 ,-1 , 0
  2274.1      .1       0    4495     .16       0  4859.1     .12       0
  4979.7     .07       0    5016     .12       0  5575.4     .16       0
  5608.3     .05       0  7097.2      .1       0    7230     .05       0
    7332     .08       0  7410.2      .1       0  8203.7     .05       0
  9271.6      .1       0
Bank Sta=4979.7,5016
XS Rating Curve= 0 ,0
Exp/Cntr=0.3,0.1
